--- Dry Comal Creek Tributary 13.prj (project) ---

Proj Title=Dry Comal Creek Tributary 13 Base Level Engineering
Current Plan=p01
Default Exp/Contr=0.3,0.1
English Units
Geom File=g01
Flow File=f01
Plan File=p01
Y Axis Title=Elevation
X Axis Title(PF)=Main Channel Distance
X Axis Title(XS)=Station
BEGIN DESCRIPTION:
Dry Comal Creek Tributary 13
END DESCRIPTION:
DSS Export Rating Curves= 0
DSS Export Rating Curve Sorted= 0
DSS Export Volume Flow Curves= 0
DXF OffsetX= 0
DXF OffsetY= 0
DXF ScaleX= 1
DXF ScaleY= 10

--- Dry Comal Creek Tributary 13.p01 (plan) ---

Plan Title=Multiple Run
Short Identifier=Multiple
Geom File=g01
Flow File=f01
Subcritical Flow
K Sum by GR= 0
Std Step Tol= 0.01
Critical Tol= 0.01
Num of Std Step Trials= 20
Max Error Tol= 0.3
Flow Tol Ratio= 0.001
Split Flow NTrial= 30
Split Flow Tol= 0.02
Split Flow Ratio= 0.02
Log Output Level= 0
Friction Slope Method= 1
Unsteady Friction Slope Method= 2
Unsteady Bridges Friction Slope Method= 1
Parabolic Critical Depth
Global Vel Dist=  1 , 1 , 1
Global Log Level= 0
CheckData=True
Encroach Param= -1, 0, 0, 0
BEGIN DESCRIPTION:
Multiple Run
END DESCRIPTION:

--- Dry Comal Creek Tributary 13.f01 (steady flow) ---

Flow Title=Multiple
Number of Profiles=7
Profile Names=10-year,25-year,50-year,1pct_min,100-year,1pct_plu,500-year
River Rch & RM= Dry Comal Creek ,Reach-1,26304
     925    1529    2089    1381    2756    5498    4745
River Rch & RM= Dry Comal Creek ,Reach-1,25022
    1262    2122    2930    1956    3903    7787    6854
River Rch & RM= Dry Comal Creek ,Reach-1,22741
    1686    2877    4012    2702    5391   10756    9641
River Rch & RM= Dry Comal Creek ,Reach-1,20478
    1863    3179    4434    2984    5953   11878   10633
River Rch & RM= Dry Comal Creek ,Reach-1,12284
    2432    4230    5975    4070    8121   16204   14871
River Rch & RM= Dry Comal Creek ,Reach-1,8232
    2750    4815    6832    4673    9323   18603   17213
River Rch & RM= Dry Comal Creek ,Reach-1,4166
    2860    5023    7141    4895    9767   19487   18108
Boundary for River Rch & Prof#=Dry Comal Creek ,Reach-1,1
Up Type=0
Dn Type=3
Dn Slope=0.005
Boundary for River Rch & Prof#=Dry Comal Creek ,Reach-1,2
Up Type=0
Dn Type=3
Dn Slope=0.005
Boundary for River Rch & Prof#=Dry Comal Creek ,Reach-1,3
Up Type=0
Dn Type=3
Dn Slope=0.005
Boundary for River Rch & Prof#=Dry Comal Creek ,Reach-1,4
Up Type=0
Dn Type=3
Dn Slope=0.005
Boundary for River Rch & Prof#=Dry Comal Creek ,Reach-1,5
Up Type=0
Dn Type=3
Dn Slope=0.005
Boundary for River Rch & Prof#=Dry Comal Creek ,Reach-1,6
Up Type=0
Dn Type=3
Dn Slope=0.005
Boundary for River Rch & Prof#=Dry Comal Creek ,Reach-1,7
Up Type=0
Dn Type=3
Dn Slope=0.005

--- Dry Comal Creek Tributary 13.g01 (geometry) ---

Geom Title=Existing Conditions
Program Version=4.10

River Reach=Dry Comal Creek ,Reach-1
Reach XY= 30
        2219525.     13805112.71      2219430.69     13804572.61
      2220045.58     13804255.42      2220117.44       13803925.
      2219578.54     13803273.53      2219524.23     13802235.69
      2219124.79     13801149.91      2219773.81     13800134.59
      2218364.94     13799264.39      2218324.56     13799009.82
      2219222.95     13797969.14      2218884.13     13797068.26
      2219481.19     13796817.19      2219623.82     13796535.48
      2218030.59     13795469.39      2217376.96     13794530.89
      2219067.14     13793381.17      2219373.98     13792814.58
       2219274.9      13791745.1      2219461.68     13791438.37
      2220445.05     13791675.21      2220814.49     13791534.81
      2220626.19      13790535.5      2221068.52     13789882.69
      2221423.54     13789878.54      2222045.01     13790325.07
      2222619.07     13789977.24      2222871.54      13790176.5
      2222822.41     13790570.03        2223675.       13790575.

Type RM Length L Ch R = 1 ,26304   ,396,396,396
BEGIN DESCRIPTION:
X18985
END DESCRIPTION:
XS GIS Cut Line= 3
      2219773.74     13805124.13      2219600.11     13805019.95
      2219059.26     13805165.56
#Sta/Elev= 30
    4691  874.47  4712.7  874.53    4740  873.67  4771.1  873.64  4856.6  872.06
  4893.4  870.76  4928.4  868.65  4933.6  868.78  4960.9  865.74  4968.4  863.95
    4990  862.81  4990.2  862.31  4993.7  862.31    4994  862.81  5002.3  862.89
  5008.3  863.96  5013.5   864.1  5023.1  865.14  5033.4  865.48  5095.5  869.73
  5147.3  871.62  5157.7  872.61  5201.4  873.72  5230.2  875.07  5261.2  875.66
  5271.6  876.25  5385.5  879.53  5426.9  881.99  5432.2  882.84  5453.6  884.78
#Mann= 3 ,-1 , 0
    4691     .12       0    4990     .05       0    4994     .12       0
Bank Sta=4990,4994
XS Rating Curve= 0 ,0
Exp/Cntr=0.3,0.1

Type RM Length L Ch R = 1 ,25908   ,440,440,440
BEGIN DESCRIPTION:
Dry Comal Creek Tributary 13 49.0
END DESCRIPTION:
XS GIS Cut Line= 3
        2219675.       13805025.        2219425.       13804675.
      2219174.97     13804725.01
#Sta/Elev= 30
  4569.8  871.96  4591.9  871.58  4598.1  871.83  4642.3  870.27  4684.1   869.8
    4705  868.48  4713.6  868.58  4778.7  867.29  4805.8  866.15  4814.4  866.31
  4820.5  865.84  4885.6   864.5  4906.5  863.55  4921.3  863.69  4927.4  863.02
    4936  863.16  4942.2  862.59  4986.4  862.14  4992.5  861.41  5018.3  861.12
  5018.6  860.62  5022.1  860.62  5022.3  861.12  5025.4  861.61  5040.7  862.44
  5081.5   865.8  5101.9  866.59  5112.1  867.43  5244.7  872.67  5254.9   872.7
#Mann= 3 ,-1 , 0
  4569.8     .12       0  5018.3     .05       0  5022.3     .12       0
Bank Sta=5018.3,5022.3
XS Rating Curve= 0 ,0
Exp/Cntr=0.3,0.1

Type RM Length L Ch R = 1 ,25468   ,446,446,446
BEGIN DESCRIPTION:
Dry Comal Creek Tributary 13 48.0
END DESCRIPTION:
XS GIS Cut Line= 3
      2220024.97     13804774.97        2219675.       13804375.
      2219374.98     13804224.99
#Sta/Elev= 30
    4473  872.23  4529.4  871.33  4551.3  870.39  4614.9  869.17  4664.2  867.56
  4678.4  866.96  4692.7  865.67  4713.6  865.41  4763.9  862.97  4819.9  862.31
  4841.7  861.53  4848.3  862.27    4891  861.97  4933.8  860.33    4948  859.25
  4962.2  857.29  4974.5  856.54  4974.7  856.04  4978.2  856.04  4978.5  856.54
  4997.3  856.97  5001.1  857.89  5012.9  858.46  5018.4  859.77  5035.2  860.71
  5040.8  861.66  5079.9  863.75  5183.4  866.73  5295.2  871.04  5339.9  872.14
#Mann= 3 ,-1 , 0
    4473     .07       0  4974.5     .05       0  4978.5     .07       0
Bank Sta=4974.5,4978.5
XS Rating Curve= 0 ,0
Exp/Cntr=0.3,0.1

Type RM Length L Ch R = 1 ,25022   ,428,428,428
BEGIN DESCRIPTION:
Dry Comal Creek Tributary 13 47.0
END DESCRIPTION:
XS GIS Cut Line= 3
      2220224.95       13804225.        2220075.       13804225.
      2219274.98       13804125.
#Sta/Elev= 30
  4846.2  869.64  4876.2  868.26  4886.2  867.41  4896.2  865.72  4921.6  863.92
  4940.8  862.54  4956.2  861.53  4986.2  858.82  4993.7  856.19  4998.7  856.19
  5006.2  853.38  5014.1  852.61  5014.4  852.11  5018.3  852.11  5018.6  852.61
  5026.4  853.75  5045.1   854.6  5086.9  857.28    5107  857.86  5248.1  860.11
  5288.4  861.58  5379.1  863.85  5469.8  865.71  5522.7   866.4  5603.3  868.52
  5631.1  870.22    5684  871.58  5731.8  873.68    5752  874.04  5802.4  875.85
#Mann= 6 ,-1 , 0
  4846.2     .12       0  4921.6     .07       0  4940.8     .12       0
  5014.1     .05       0  5018.6     .12       0  5045.1     .07       0
Bank Sta=5014.1,5018.6
XS Rating Curve= 0 ,0
Exp/Cntr=0.3,0.1

Type RM Length L Ch R = 1 ,24594   ,446,446,446
BEGIN DESCRIPTION:
Dry Comal Creek Tributary 13 46.0
END DESCRIPTION:
XS GIS Cut Line= 3
      2220225.02       13803825.        2220075.       13803825.
      2219525.04     13803924.99
#Sta/Elev= 30
    4850  869.74    4890  867.64    4900  866.77    4910  865.15    4920  863.92
    4930  862.11    4940  859.92    4950  858.24    4960  855.57    4970  851.37
  4977.8  849.94  4978.1  849.44    4982  849.44  4982.3  849.94    4990  850.81
  5002.6  850.64  5031.8  852.47  5050.8  853.98  5091.5  855.59  5152.5  857.01
  5213.5  857.42  5255.4  858.48  5308.8   859.4  5376.1  861.51  5415.5   862.1
  5437.1  863.18  5457.4  863.78    5479  864.93  5536.7  866.77    5559  867.42
#Mann= 4 ,-1 , 0
    4850     .12       0  4977.8     .05       0  4982.3     .12       0
  5536.7    .035       0
Bank Sta=4977.8,4982.3
XS Rating Curve= 0 ,0
Exp/Cntr=0.3,0.1

Type RM Length L Ch R = 1 ,24148   ,475,475,475
BEGIN DESCRIPTION:
Dry Comal Creek Tributary 13 45.0
END DESCRIPTION:
XS GIS Cut Line= 3
      2220225.03       13803475.        2219825.       13803475.
      2219475.03     13803574.99
#Sta/Elev= 30
  4600.3  868.89  4630.3  867.49  4650.3  865.84  4680.3   864.8  4710.3  863.44
  4720.3  862.68  4810.3  859.16  4860.3  857.85  4890.3  855.39  4950.3  851.81
  4980.3  849.41  4997.8  848.81  5010.7  849.01  5014.9  848.77  5015.3  848.27
  5019.2  848.27  5019.5  848.77  5031.5  849.42  5083.5  850.38  5114.7  851.97
  5135.5  853.95  5145.9  854.58  5177.1  856.41  5218.7  858.12  5235.6  859.47
  5260.3  860.15  5291.5  862.19  5313.6  862.75  5322.7  863.52  5364.3  864.82
#Mann= 3 ,-1 , 0
  4600.3     .12       0  5014.9     .05       0  5019.5     .12       0
Bank Sta=5014.9,5019.5
XS Rating Curve= 0 ,0
Exp/Cntr=0.3,0.1

Type RM Length L Ch R = 1 ,23673   ,449,449,449
BEGIN DESCRIPTION:
Dry Comal Creek Tributary 13 44.0
END DESCRIPTION:
XS GIS Cut Line= 3
      2220324.95     13803274.99        2219575.       13803125.
      2219375.01     13803224.99
#Sta/Elev= 30
  4231.1  869.77  4251.4  869.73  4261.6  868.34    4282  867.27  4394.2  863.06
  4414.6   861.5  4445.2  860.86  4465.6  859.37  4506.4  858.75  4598.2  855.73
  4618.6  855.96  4659.4  854.78  4761.3  853.74  4904.1   850.6  4955.1  848.29
  4965.3  846.86  4998.7  845.13    5016  843.32  5016.3  842.82  5020.3  842.82
  5020.6  843.32  5032.2  844.42  5040.6  846.64    5049  847.95  5054.6  848.04
  5071.4  850.08  5093.7  851.92  5121.7  852.88  5183.2  858.71  5219.5  860.58
#Mann= 3 ,-1 , 0
  4231.1     .12       0    5016     .05       0  5020.6     .12       0
Bank Sta=5016,5020.6
XS Rating Curve= 0 ,0
Exp/Cntr=0.3,0.1

Type RM Length L Ch R = 1 ,23224   ,483,483,483
BEGIN DESCRIPTION:
Dry Comal Creek Tributary 13 43.0
END DESCRIPTION:
XS GIS Cut Line= 3
      2219824.99       13802525.        2219425.       13802725.
      2219225.01       13802825.
#Sta/Elev= 30
  4552.7  858.13  4583.4  857.75  4619.8  855.39  4664.5  853.56  4686.9  851.62
  4709.2  850.72  4717.6  850.55  4723.2  851.02    4740  850.28  4767.9  850.13
  4812.6  848.99  4879.7  846.57  4896.5  845.39  4924.4   844.9  4985.9  842.14
  4991.5  841.53  4994.3  840.67  4994.8  840.17  4999.5  840.17  4999.9  840.67
  5013.9  841.32  5027.9  845.19  5030.6  846.64    5053  849.55  5058.6  849.36
  5089.3  850.58  5120.1  852.81  5178.8  855.13  5209.5  857.52  5223.5  857.74
#Mann= 3 ,-1 , 0
  4552.7     .12       0  4994.3     .05       0  4999.9     .12       0
Bank Sta=4994.3,4999.9
XS Rating Curve= 0 ,0
Exp/Cntr=0.3,0.1

Type RM Length L Ch R = 1 ,22741   ,446,446,446
BEGIN DESCRIPTION:
Dry Comal Creek Tributary 13 42.0
END DESCRIPTION:
XS GIS Cut Line= 3
      2219674.97     13802225.01        2219525.       13802275.
      2218975.02     13802075.01
#Sta/Elev= 30
  4838.1  855.74  4859.1  854.83  4869.7  854.98  4911.9  850.85    4954  850.06
  4964.6  848.47  4985.6  842.93  4993.5  840.01  4998.8  840.01  5006.2   838.5
  5013.7  838.16  5014.2  837.66  5020.7  837.66  5021.2  838.16  5042.1  838.31
  5072.7  840.03  5081.3  841.14  5134.5  843.39  5166.4   844.4  5262.2   845.7
    5326  848.16  5362.6  848.61  5540.8  855.26  5543.1  855.95  5549.5  857.87
  5560.1  862.23  5566.1  862.73  5571.4  861.56  5578.8   858.2  5581.4   858.2
#Mann= 4 ,-1 , 0
  4838.1     .12       0  5013.7     .05       0  5021.2     .12       0
  5543.1    .035       0
Bank Sta=5013.7,5021.2
XS Rating Curve= 0 ,0
Exp/Cntr=0.3,0.1

Type RM Length L Ch R = 1 ,22295   ,451,451,451
BEGIN DESCRIPTION:
Dry Comal Creek Tributary 13 41.0
END DESCRIPTION:
XS GIS Cut Line= 3
      2219574.98       13801875.        2219375.       13801875.
      2218974.98     13802025.01
#Sta/Elev= 30
  4795.5  853.07  4905.5  845.17  4955.5     840  4965.5  837.54  4975.5  835.71
  5001.5  834.83    5002  834.33  5008.5  834.33    5009  834.83  5016.8  835.86
  5027.5  836.34  5035.5   837.7  5065.8  839.86  5096.1  840.92  5126.3  842.79
    5145  844.29  5151.2  845.32  5156.6  844.38  5176.2  845.38  5181.5  845.24
  5219.8  848.24  5275.3  849.96  5322.1  852.75  5369.3  854.74  5381.7   858.7
  5390.6   863.2  5401.3  863.29  5407.6  860.24  5412.9  858.81  5422.7  858.16
#Mann= 5 ,-1 , 0
  4795.5     .12       0  5001.5     .05       0    5009     .12       0
  5275.3    .035       0  5381.7     .12       0
Bank Sta=5001.5,5009
XS Rating Curve= 0 ,0
Exp/Cntr=0.3,0.1

Type RM Length L Ch R = 1 ,21844   ,450,450,450
BEGIN DESCRIPTION:
Dry Comal Creek Tributary 13 40.0
END DESCRIPTION:
XS GIS Cut Line= 3
      2219625.01       13801625.        2219225.       13801475.
      2218825.01       13801325.
#Sta/Elev= 30
  4567.1   853.2  4582.2  852.99  4637.4  849.99  4697.9  848.27    4778  843.04
  4838.6  841.49  4863.5  840.03  4899.1  839.02  4918.7  837.05  4948.9  835.13
  4962.3  835.42  4972.9  834.61  5011.9  834.36  5012.4  833.86    5019  833.86
  5019.5  834.36  5034.4  835.49  5039.7  834.96  5064.6  838.56    5070  837.84
  5079.7  838.74  5125.1   839.5  5143.8  840.66    5175   843.8  5180.3  843.86
  5218.6  848.84  5290.7  853.54  5326.3  855.22  5376.1   861.5  5421.5  863.97
#Mann= 3 ,-1 , 0
  4567.1     .12       0  5011.9     .05       0  5019.5     .12       0
Bank Sta=5011.9,5019.5
XS Rating Curve= 0 ,0
Exp/Cntr=0.3,0.1

Type RM Length L Ch R = 1 ,21394   ,469,469,469
BEGIN DESCRIPTION:
Dry Comal Creek Tributary 13 39.0
END DESCRIPTION:
XS GIS Cut Line= 4
      2219759.83     13801367.17        2219175.       13801075.
        2219075.       13801075.      2218963.25       13801075.
#Sta/Elev= 30
  4341.2   849.4  4360.3  849.42    4405  847.96  4511.3     846  4645.5  844.39
    4682  842.48  4740.5  840.44  4757.3   838.7  4762.9  838.82  4779.7  836.21
  4793.7  835.85  4891.5  837.52  4927.9  836.98  4950.2  835.91  4964.2  834.37
    4981  830.67  4997.5  830.21  5001.2  829.46  5001.7  828.96  5008.3  828.96
  5008.8  829.46    5015  830.23    5025  834.26    5035  839.97    5045  843.28
    5065  845.63    5085  849.24    5125  852.63    5195  857.48  5206.7  857.57
#Mann= 3 ,-1 , 0
  4341.2     .12       0  5001.2     .05       0  5008.8     .12       0
Bank Sta=5001.2,5008.8
XS Rating Curve= 0 ,0
Exp/Cntr=0.3,0.1

Type RM Length L Ch R = 1 ,20925   ,447,447,447
BEGIN DESCRIPTION:
Dry Comal Creek Tributary 13 38.0
END DESCRIPTION:
XS GIS Cut Line= 4
      2219825.01       13800725.        2219375.       13800675.
        2219175.       13800675.      2219048.88       13800675.
#Sta/Elev= 30
  4547.2  844.35  4627.7  842.22  4657.9   840.9  4738.5  835.65  4748.4  836.06
  4818.9  834.42    4839  832.42  4879.2  833.34  4899.4  833.03  4949.7  830.72
  4959.7  829.61  4979.9   830.8  4986.1  828.89  4986.6  828.39  4993.3  828.39
  4993.8  828.89  4997.5  829.69    5020  829.48    5030  830.49    5040   832.3
    5050  835.79    5060  837.74    5080  839.29    5140  841.85    5160  844.16
    5190  844.84  5197.5   845.9    5240  848.16    5250  849.16  5326.1  851.34
#Mann= 4 ,-1 , 0
  4547.2    .035       0  4738.5     .12       0  4986.1     .05       0
  4993.8     .12       0
Bank Sta=4986.1,4993.8
XS Rating Curve= 0 ,0
Exp/Cntr=0.3,0.1

Type RM Length L Ch R = 1 ,20478   ,428,428,428
BEGIN DESCRIPTION:
Dry Comal Creek Tributary 13 37.0
END DESCRIPTION:
XS GIS Cut Line= 3
        2219975.       13800175.        2219675.       13800375.
      2219124.97     13800475.01
#Sta/Elev= 30
  4639.6  859.72  4704.2  853.45  4740.3  847.88  4755.3   843.9  4791.3  839.35
  4848.4  836.25  4863.4  834.24  4869.4  834.98  4878.5  833.43  4884.5   834.1
  4899.5  830.63  4905.7   832.2  4914.5  830.37  4920.5   831.9  4935.6  826.78
  4941.6  828.59  4950.6  826.92  4956.6  828.18  4964.6  826.95  4982.6  826.56
  4983.1  826.06  4990.7  826.56  4992.6  827.94  5002.7  827.26  5026.8  829.24
  5122.8  830.25  5152.6  830.25  5223.5  833.66  5424.8  841.51  5559.2  846.34
#Mann= 8 ,-1 , 0
  4639.6     .12       0  4905.7     .07       0  4964.6     .12       0
  4982.6     .05       0  4990.7     .12       0  5122.8     .07       0
  5223.5    .035       0  5424.8     .12       0
Bank Sta=4982.6,4990.7
XS Rating Curve= 0 ,0
Exp/Cntr=0.3,0.1

Type RM Length L Ch R = 1 ,20050   ,469,469,469
BEGIN DESCRIPTION:
Dry Comal Creek Tributary 13 36.0
END DESCRIPTION:
XS GIS Cut Line= 4
      2219775.02     13799974.99        2219675.       13800025.
        2219325.       13800275.      2219099.06     13800436.39
#Sta/Elev= 30
  4888.2  851.56    4919  848.56  4924.6  847.59  4941.3   842.6  4946.9  839.78
  4963.7  833.05  4969.3  828.47    4982  822.64  4982.5  822.14  4989.6  822.14
  4990.1  822.64  4997.2  823.27  5007.4  823.25  5013.8  824.56  5022.1  826.37
  5036.9  826.47  5049.2  827.85  5057.8   827.5    5086  827.88    5096  828.95
  5114.3  829.54  5137.5  831.07  5221.2  833.85  5258.5  834.23  5261.2  834.24
  5286.4  834.17  5315.9  835.58  5384.9  836.57  5508.6  840.18  5707.8   845.9
#Mann= 10 ,-1 , 0
  4888.2     .12       0    4982     .05       0  4990.1     .12       0
  5013.8      .1       0    5096    .035       0  5137.5     .07       0
  5258.5    .035       0  5261.2     .12       0  5384.9     .07       0
  5508.6     .12       0
Bank Sta=4982,4990.1
XS Rating Curve= 0 ,0
Exp/Cntr=0.3,0.1

Type RM Length L Ch R = 1 ,19581   ,466,466,466
BEGIN DESCRIPTION:
Dry Comal Creek Tributary 13 35.0
END DESCRIPTION:
XS GIS Cut Line= 4
      2219424.96     13799675.02        2219325.       13799725.
        2219125.       13800125.      2219079.19     13800216.61
#Sta/Elev= 30
  4888.5  838.75  4888.7  838.75  4896.8  837.95  4919.2  836.65  4941.6  833.89
  4955.5  831.47  4963.9  829.44  4969.5  827.15  4986.3  824.15  4991.9  822.19
  5003.1  821.88  5004.5  821.24    5005  820.74  5012.2  820.74  5012.7  821.24
  5022.6  822.25  5036.6   824.9    5045   825.3    5058  824.93  5098.1  826.66
    5126  828.86  5165.2  830.47  5215.5  832.13  5274.8   832.9  5313.3  833.65
  5397.6  836.82  5433.5  838.83  5450.3  838.98  5483.8  840.42  5549.9  841.98
#Mann= 7 ,-1 , 0
  4888.5     .12       0  4888.7      .1       0  5004.5     .05       0
  5012.7      .1       0    5058     .12       0  5274.8     .07       0
  5397.6    .035       0
Bank Sta=5004.5,5012.7
XS Rating Curve= 0 ,0
Exp/Cntr=0.3,0.1

Type RM Length L Ch R = 1 ,19115   ,480,480,480
BEGIN DESCRIPTION:
Dry Comal Creek Tributary 13 34.0
END DESCRIPTION:
XS GIS Cut Line= 4
      2219224.96     13799375.02        2218925.       13799525.
        2218775.       13799875.      2218742.44     13799950.96
#Sta/Elev= 30
    4671   837.6  4701.7  836.74  4782.8  831.86  4805.1  829.92  4827.5  826.83
  4849.8  825.12  4872.2  824.22  4925.3  824.48  4947.7  823.63  4953.3  822.44
  4992.4  822.08  4993.8  821.23  4994.3  820.73  5001.6  820.73  5002.1  821.23
  5009.1  821.29  5015.4  822.17  5020.9  821.94  5028.1   823.3  5049.9  825.42
    5068  826.92  5082.5  827.49    5097  827.38  5136.9  828.78  5220.3  830.24
  5301.9  833.28  5320.1   834.9  5325.5  834.62  5430.7  838.67  5469.8  839.35
#Mann= 3 ,-1 , 0
    4671     .12       0  4993.8     .05       0  5002.1     .12       0
Bank Sta=4993.8,5002.1
XS Rating Curve= 0 ,0
Exp/Cntr=0.3,0.1

Type RM Length L Ch R = 1 ,18635   ,482,482,482
BEGIN DESCRIPTION:
Dry Comal Creek Tributary 13 33.0
END DESCRIPTION:
XS GIS Cut Line= 4
        2219075.       13799075.        2218525.       13799325.
        2218325.       13799425.       2218230.6      13799472.2
#Sta/Elev= 30
  4395.1  835.42    4450   834.5  4515.9  829.81  4537.9  828.97  4636.8  827.82
  4771.9  827.97  4887.2   826.2  4915.8  825.12  4933.3  823.79  4944.3  820.73
    4973   818.2  4973.5   817.7    4981   817.7  4981.5   818.2  5007.6  818.26
  5013.2   819.1    5030  819.04  5066.3  820.93  5088.7  820.25  5133.4  821.17
  5141.8  822.07  5155.8  825.23  5178.1  833.51  5186.5  836.18  5192.1   836.9
  5220.1  838.78  5259.2  839.54  5289.9   841.1  5320.7  843.46  5328.4  843.24
#Mann= 3 ,-1 , 0
  4395.1     .12       0    4973     .05       0  4981.5     .12       0
Bank Sta=4973,4981.5
XS Rating Curve= 0 ,0
Exp/Cntr=0.3,0.1

Type RM Length L Ch R = 1 ,18153   ,466,466,466
BEGIN DESCRIPTION:
Dry Comal Creek Tributary 13 32.0
END DESCRIPTION:
XS GIS Cut Line= 4
        2219025.       13799025.        2218325.       13798975.
        2218225.       13798975.      2218101.78       13798975.
#Sta/Elev= 30
  4302.6  834.62  4342.7  832.99  4370.3  830.87  4392.8  830.08  4432.9  827.71
    4453  827.24  4503.1  827.04  4623.4  825.69    4651  825.68    4656  826.02
  4673.5   825.4  4796.4  824.85    4844  822.35  4904.1  820.35  4914.2  820.41
  4954.3  815.52    4980   814.3  4980.5   813.8  4988.1   813.8  4988.6   814.3
  4994.4   815.5  5001.9  817.98  5006.9  817.98  5014.4   823.8  5034.4  837.86
  5044.4  839.59  5074.4  842.03  5134.4  844.44  5204.4  848.75  5227.6  849.51
#Mann= 3 ,-1 , 0
  4302.6     .12       0    4980     .05       0  4988.6     .12       0
Bank Sta=4980,4988.6
XS Rating Curve= 0 ,0
Exp/Cntr=0.3,0.1

Type RM Length L Ch R = 1 ,17687   ,469,469,469
BEGIN DESCRIPTION:
Dry Comal Creek Tributary 13 31.0
END DESCRIPTION:
XS GIS Cut Line= 5
      2218983.58     13798880.72        2218825.       13798775.
        2218525.       13798575.        2218425.       13798525.
      2218304.65     13798464.83
#Sta/Elev= 30
  4453.3  832.66  4558.3  830.31  4621.4  829.58  4640.9   828.8  4657.4  829.05
  4679.9  828.34  4708.5  826.64  4765.6  825.03  4801.6  822.13  4824.2  821.63
  4852.7  819.86  4924.8  817.92  4968.4  814.11  4975.9  814.18  4986.6  812.41
  4987.1  811.91  4994.8  811.91  4995.3  812.41  5001.4  814.28  5007.2  814.28
  5012.8  816.53  5018.4  820.56  5026.8   824.9  5057.6  831.02  5093.9  834.24
    5119  834.98    5147  837.44  5169.4  838.79  5219.7  839.41  5250.8  840.37
#Mann= 3 ,-1 , 0
  4453.3     .12       0  4986.6     .05       0  4995.3     .12       0
Bank Sta=4986.6,4995.3
XS Rating Curve= 0 ,0
Exp/Cntr=0.3,0.1

Type RM Length L Ch R = 1 ,17218   ,466,466,466
BEGIN DESCRIPTION:
Dry Comal Creek Tributary 13 30.0
END DESCRIPTION:
XS GIS Cut Line= 5
      2219142.51     13798676.26        2219075.       13798575.
        2218875.       13798275.        2218725.       13798225.
       2218574.6     13798174.87
#Sta/Elev= 30
  4517.5   830.3  4523.5  829.75  4589.6  828.39  4595.6  828.55  4616.7  827.53
  4642.2  827.13  4697.8  825.26  4711.3  824.39  4790.9   821.2    4812  820.83
  4941.2  814.22  4950.2  815.42  4956.2  813.98  4963.7  812.87  4992.4  811.37
  4992.9  810.87  5000.6  810.87  5001.1  811.37  5010.3   811.8  5041.9  817.33
  5052.5  820.98  5073.5  822.55  5084.1  824.78  5115.7  827.46  5136.8  828.66
  5160.5  829.07  5178.9  830.34    5200  831.05  5252.7  831.36  5316.4  832.67
#Mann= 3 ,-1 , 0
  4517.5     .12       0  4992.4     .05       0  5001.1     .12       0
Bank Sta=4992.4,5001.1
XS Rating Curve= 0 ,0
Exp/Cntr=0.3,0.1

Type RM Length L Ch R = 1 ,16752   ,457,457,457
BEGIN DESCRIPTION:
Dry Comal Creek Tributary 13 29.0
END DESCRIPTION:
XS GIS Cut Line= 5
      2219495.92     13798110.46        2219325.       13798025.
        2219225.       13797975.        2218725.       13798075.
      2218638.31     13798092.34
#Sta/Elev= 30
  4692.3  827.17  4752.8  826.14  4793.9  825.49  4886.2  825.08  4919.7  824.12
  4942.1   822.5  4958.9  820.36  4964.4  820.25  4972.8  819.26  4986.8  815.77
  4992.4  811.45  4997.7  811.45    5001  809.05  5001.5  808.55  5009.3  808.55
  5009.8  809.05    5036  811.64  5066.6  811.46  5127.8  814.49  5148.2  816.37
  5199.2  818.55  5270.5  819.37  5372.5  821.79  5382.7  822.98  5392.9   822.6
  5403.1  822.98  5454.1  825.01  5484.7  826.87  5525.5  827.24  5593.5  829.54
#Mann= 4 ,-1 , 0
  4692.3    .035       0  4752.8     .12       0    5001     .05       0
  5009.8     .12       0
Bank Sta=5001,5009.8
XS Rating Curve= 0 ,0
Exp/Cntr=0.3,0.1

Type RM Length L Ch R = 1 ,16295   ,418,418,418
BEGIN DESCRIPTION:
Dry Comal Creek Tributary 13 28.0
END DESCRIPTION:
XS GIS Cut Line= 3
      2219475.05     13797725.02        2219075.       13797575.
      2218674.97     13797775.02
#Sta/Elev= 30
  4572.4   822.9    4603  822.46    4612  822.84  4674.3  822.53  4753.1  821.98
  4838.6  819.97  4874.2  818.44  4882.2  817.84  4899.1  814.74  4904.4  816.05
    4924   809.9  4929.3   810.7  4935.6  807.75  4941.8   807.6  4942.3   807.1
  4950.1   807.1  4950.6   807.6  4978.3  808.35    5008  807.75    5022  808.85
    5036  811.46  5066.7  813.26  5080.7  812.86  5103.1  813.76    5268  816.22
  5312.7  818.62  5326.7  818.51  5357.4   819.9  5379.8   821.5  5446.9  823.41
#Mann= 6 ,-1 , 0
  4572.4    .035       0    4603     .07       0    4612    .035       0
  4674.3     .12       0  4941.8     .05       0  4950.6     .12       0
Bank Sta=4941.8,4950.6
XS Rating Curve= 0 ,0
Exp/Cntr=0.3,0.1

Type RM Length L Ch R = 1 ,15877   ,448,448,448
BEGIN DESCRIPTION:
Dry Comal Creek Tributary 13 27.0
END DESCRIPTION:
XS GIS Cut Line= 3
      2220025.01       13797925.        2218925.       13797225.
      2218525.04     13797524.97
#Sta/Elev= 30
  3704.7  823.56  3707.5  823.56  3890.3  821.87  3921.4  820.48  3936.7  821.17
  3957.9  820.46  4051.2  820.72  4082.7  821.43  4165.8  821.01  4275.1   821.3
  4464.2  820.79  4630.9  817.14    4653  817.59  4747.8  813.04    4807  812.04
  4842.6  813.05    4901  810.75  4906.9  811.48  4922.2  809.11  4990.6  807.11
  4991.1  806.61  4999.4  807.11  5036.7  809.24  5072.1  809.05  5151.3  810.75
    5195  814.55  5215.8  815.28  5330.4  816.64  5401.3  820.31  5508.5  822.68
#Mann= 10 ,-1 , 0
  3704.7    .063       0  3707.5    .035       0  3890.3     .12       0
  3936.7     .07       0  4051.2    .035       0  4082.7     .12       0
  4165.8    .035       0  4275.1     .12       0  4990.6     .05       0
  4999.4     .12       0
Bank Sta=4990.6,4999.4
XS Rating Curve= 0 ,0
Exp/Cntr=0.3,0.1

Type RM Length L Ch R = 1 ,15429   ,483,483,483
BEGIN DESCRIPTION:
Dry Comal Creek Tributary 13 26.0
END DESCRIPTION:
XS GIS Cut Line= 3
      2219374.99     13797324.99        2219075.       13796875.
      2218585.35     13796795.99
#Sta/Elev= 30
  4463.6  817.75  4535.7  815.53  4621.3  811.53  4674.7   810.6  4723.5   809.7
  4780.6  809.75  4831.7   808.7  4909.8  808.26  4918.8  807.63  4924.8  807.87
  4939.8  806.05  4945.8  805.85  4960.8  803.54  4968.4  803.41  4975.9  802.44
    4997  802.26  4997.5  801.76  5005.4  801.76  5005.9  802.26  5024.7  803.34
  5032.8   805.3  5037.8  807.85  5044.9  808.69  5055.1   810.8  5099.6  815.87
  5146.2  817.34  5208.9   818.2  5351.8  818.75  5475.4  818.31  5500.4  817.92
#Mann= 6 ,-1 , 0
  4463.6    .035       0  4674.7     .12       0    4997     .05       0
  5005.9     .12       0  5208.9     .07       0  5475.4     .12       0
Bank Sta=4997,5005.9
XS Rating Curve= 0 ,0
Exp/Cntr=0.3,0.1

Type RM Length L Ch R = 1 ,14946   ,441,441,441
BEGIN DESCRIPTION:
Dry Comal Creek Tributary 13 25.0
END DESCRIPTION:
XS GIS Cut Line= 3
      2220004.58     13796991.28        2219525.       13796775.
      2218974.98       13796625.
#Sta/Elev= 30
  4474.2  825.75  4682.2  820.27  4766.8  816.26  4772.3  816.67  4802.8  815.72
  4818.6  814.63  4841.7  811.76  4847.2  812.11    4888  809.45  4893.5   809.9
  4916.6  807.69  4939.7  804.77  4956.4  801.68  4963.9   799.1  4964.4   798.6
  4972.3   798.6  4972.8   799.1  4984.8  800.03  5041.8  802.55    5097  802.29
  5145.4  804.81  5166.1   804.8  5205.9  807.29    5218   808.7  5290.5  811.28
  5364.6   812.8  5433.9  814.35  5478.8  814.36  5525.1  815.32  5570.4  815.29
#Mann= 6 ,-1 , 0
  4474.2     .12       0  4963.9     .05       0  4972.8     .12       0
  4984.8     .07       0  5364.6    .035       0  5525.1     .07       0
Bank Sta=4963.9,4972.8
XS Rating Curve= 0 ,0
Exp/Cntr=0.3,0.1

Type RM Length L Ch R = 1 ,14505   ,451,451,451
BEGIN DESCRIPTION:
Dry Comal Creek Tributary 13 24.0
END DESCRIPTION:
XS GIS Cut Line= 3
       2219939.5     13796191.83        2219525.       13796425.
      2219080.18     13796574.62
#Sta/Elev= 30
  4530.6  831.46  4587.7  829.47  4593.5  828.25  4631.1  826.47    4662  826.87
  4690.4  824.73  4706.3  824.98    4793   820.5  4830.6  819.66  4889.9  816.54
  4911.5  814.97  4917.3  813.58  4933.2  814.43  4938.9  812.65  4948.8  813.54
  4954.9  810.64  4960.6  803.39  4970.8   797.2  4976.5  793.97  4987.9  790.19
  4988.4  789.69  4997.1  790.19  4998.2  792.88  5003.3  795.99  5048.2  799.56
  5090.6  804.38  5227.7  811.93  5267.7  812.35  5368.5  811.91  5475.5  813.53
#Mann= 4 ,-1 , 0
  4530.6     .12       0  4987.9     .05       0  4997.1     .12       0
  5267.7    .035       0
Bank Sta=4987.9,4997.1
XS Rating Curve= 0 ,0
Exp/Cntr=0.3,0.1

Type RM Length L Ch R = 1 ,14054   ,469,469,469
BEGIN DESCRIPTION:
Dry Comal Creek Tributary 13 23.0
END DESCRIPTION:
XS GIS Cut Line= 3
      2219452.56     13795837.63        2219175.       13796175.
      2218931.72     13796504.31
#Sta/Elev= 30
  4558.6  831.94    4583  830.31  4590.8  830.44  4632.9  828.17  4640.3  827.28
  4747.2  823.93  4768.1   822.4  4796.7   821.5  4803.2  820.62  4846.3  817.89
    4853  817.97  4874.9  816.21  4910.1  811.69  4938.8  805.79  4953.1  801.47
  4959.6  800.21  4967.5  797.61  4992.2  792.89  5004.4  792.43  5004.9  791.93
  5013.2  791.93  5013.7  792.43  5059.1  795.72    5103  800.01  5181.9  803.96
  5238.7   807.4  5274.2  808.24  5303.4  809.87  5385.3  812.77  5404.9  813.15
#Mann= 5 ,-1 , 0
  4558.6     .12       0  5004.4     .05       0  5013.7     .12       0
  5181.9     .07       0  5385.3    .035       0
Bank Sta=5004.4,5013.7
XS Rating Curve= 0 ,0
Exp/Cntr=0.3,0.1

Type RM Length L Ch R = 1 ,13585   ,442,442,442
BEGIN DESCRIPTION:
Dry Comal Creek Tributary 13 22.0
END DESCRIPTION:
XS GIS Cut Line= 3
      2218925.03     13795874.98        2218775.       13795975.
      2218574.98     13796225.02
#Sta/Elev= 30
  4819.7  806.44  4855.8  804.32  4863.3  802.63  4884.3  800.87  4899.4  800.83
  4914.4  799.77  4927.9  798.05  4935.4  796.63  4941.4  794.77  4950.4  794.32
  4956.4  791.12    4964  790.06  4977.5  789.79  4987.8   788.7  4988.3   788.2
  4996.7   788.2  4997.2   788.7  5007.2  790.38    5028   792.1    5036   793.3
    5064  795.09  5077.7  795.21  5085.7  796.03  5120.9  796.62  5170.5  798.53
  5192.1  800.42  5234.5  802.54  5256.1  805.59  5277.7  807.73  5320.2   809.4
#Mann= 3 ,-1 , 0
  4819.7     .12       0  4987.8     .05       0  4997.2     .12       0
Bank Sta=4987.8,4997.2
XS Rating Curve= 0 ,0
Exp/Cntr=0.3,0.1

Type RM Length L Ch R = 1 ,13143   ,446,446,446
BEGIN DESCRIPTION:
Dry Comal Creek Tributary 13 21.0
END DESCRIPTION:
XS GIS Cut Line= 3
      2218575.04     13795624.98        2218425.       13795725.
      2218275.01     13796024.97
#Sta/Elev= 30
  4825.4  806.26    4848  804.34    4869  803.47  4905.1  799.81  4920.1  797.02
  4926.1  794.96  4933.6   793.4  4947.1  791.64  4977.2  790.73  4983.2  789.86
  4998.2  789.24  5019.7  791.04  5028.1  792.74  5050.4  795.67  5072.8  795.92
  5153.9  791.66    5193  787.08  5198.6  785.32  5210.7  783.43  5211.2  782.93
  5219.6  782.93  5220.1  783.43  5220.9  786.83  5237.7   793.8  5243.3  798.06
  5251.7   801.8  5265.7     805    5288  806.55  5310.4  809.93  5341.1  810.42
#Mann= 3 ,-1 , 0
  4825.4     .12       0  5210.7     .05       0  5220.1     .12       0
Bank Sta=5210.7,5220.1
XS Rating Curve= 0 ,0
Exp/Cntr=0.3,0.1

Type RM Length L Ch R = 1 ,12697   ,413,413,413
BEGIN DESCRIPTION:
Dry Comal Creek Tributary 13 20.0
END DESCRIPTION:
XS GIS Cut Line= 3
      2218322.36      13795256.9        2218075.       13795475.
      2217944.72     13795647.56
#Sta/Elev= 30
  4665.4  811.12  4789.8  803.81  4824.9   802.3  4867.6  798.05  4888.5  794.76
  4924.5  790.55  4959.6  783.97  4967.2   780.9  4973.8  779.37  4988.1  774.34
  4991.8   770.9  4998.3   770.9  5002.5  769.17    5004  769.05  5004.5  768.55
    5013  768.55  5013.5  769.05    5017  771.29  5023.3  772.81  5031.6   775.9
  5037.9  779.66  5052.4  785.87  5058.7  789.58    5067   792.4  5081.5  794.16
  5095.4  794.84  5131.5  797.81  5137.8  797.73  5181.4     800  5211.4  800.56
#Mann= 3 ,-1 , 0
  4665.4     .12       0    5004     .05       0  5013.5     .12       0
Bank Sta=5004,5013.5
XS Rating Curve= 0 ,0
Exp/Cntr=0.3,0.1

Type RM Length L Ch R = 1 ,12284   ,246,246,246
BEGIN DESCRIPTION:
Dry Comal Creek Tributary 13 19.0
END DESCRIPTION:
XS GIS Cut Line= 3
      2217973.38     13795009.52        2217825.       13795175.
      2217559.61     13795293.25
#Sta/Elev= 30
  4777.7  801.81    4809  799.83  4844.1  798.77  4851.6  797.58  4858.3   797.7
  4872.5  794.85  4879.2  795.67  4886.7  795.11  4893.4  795.62  4921.8  793.06
  4929.3  790.83    4936  786.17  4943.5  779.65  4950.2   772.6  4964.4  768.62
  4980.1  767.24  4980.6  766.74  4991.6  766.74  4992.1  767.24  4996.6   768.7
  5002.7   768.7  5032.1  774.83  5043.7  779.05  5054.7  780.96  5060.8  783.39
  5089.5   787.9  5130.5  789.05  5182.4   792.5  5257.6  803.74  5290.5  806.22
#Mann= 3 ,-1 , 0
  4777.7     .12       0  4980.1     .05       0  4992.1     .12       0
Bank Sta=4980.1,4992.1
XS Rating Curve= 0 ,0
Exp/Cntr=0.3,0.1

Type RM Length L Ch R = 1 ,12038   ,224,224,224
BEGIN DESCRIPTION:
X18984
END DESCRIPTION:
XS GIS Cut Line= 2
      2217810.27     13794852.78      2217502.93     13795169.87
#Sta/Elev= 30
  4818.2   797.2  4851.7  796.09  4901.3  792.72  4915.5  791.39  4943.8  787.23
  4957.9  783.12  4972.1  776.92    4979  771.39  4986.2  767.34  4993.2   766.6
  4994.4     765  4994.9   764.5  5005.9   764.5  5006.4     765  5014.5  765.06
  5021.5  766.36  5028.7  765.87  5035.6  766.85  5042.8  769.36  5049.8   772.9
  5063.9  777.99  5078.1  781.65  5092.2  783.96  5106.4  785.44    5163  789.08
  5169.9  789.12  5191.3  791.41  5212.4  792.82  5247.8  798.56  5259.8  798.45
#Mann= 3 ,-1 , 0
  4818.2     .12       0  4994.4     .05       0  5006.4     .12       0
Bank Sta=4994.4,5006.4
XS Rating Curve= 0 ,0
Exp/Cntr=0.3,0.1

Type RM Length L Ch R = 1 ,11814   ,243,243,243
BEGIN DESCRIPTION:
Dry Comal Creek Tributary 13 18.0
END DESCRIPTION:
XS GIS Cut Line= 3
      2217624.97     13794775.01        2217525.       13794825.
      2217374.99       13794875.
#Sta/Elev= 30
  4888.2  787.95  4896.6  787.85  4902.1  787.21  4916.1  786.74  4924.5  785.94
  4932.9  784.35  4941.3  781.99  4946.9  777.99  4955.3  773.18  4963.6   766.4
  4969.2  765.34  4977.6  763.14  4979.9  761.66  4980.4  761.16  4991.5  761.16
    4992  761.66  4997.2  762.32  5002.6  762.32  5010.5  762.88  5021.1  766.36
  5042.1  771.18  5052.7  776.27  5073.8  782.75  5084.3  788.72  5094.8   792.3
  5105.4  795.39  5115.9  798.96    5137  802.64  5155.5  806.62  5158.1  806.62
#Mann= 3 ,-1 , 0
  4888.2     .12       0  4979.9     .05       0    4992     .12       0
Bank Sta=4979.9,4992
XS Rating Curve= 0 ,0
Exp/Cntr=0.3,0.1

Type RM Length L Ch R = 1 ,11571   ,180,180,180
BEGIN DESCRIPTION:
X18981
END DESCRIPTION:
XS GIS Cut Line= 2
      2217676.73     13794636.86      2217165.75     13794632.04
#Sta/Elev= 30
  4708.6  790.01  4730.3  789.48  4750.3  789.33  4760.3   788.9  4790.3  788.68
  4830.3  787.57  4860.3  785.71  4870.3  784.42  4890.3  780.29  4920.3   772.7
  4930.3  769.02  4940.3  766.04  4960.3  763.89  4970.3  760.93  4984.3  758.12
  4984.8  757.62  4995.9  757.62  4996.4  758.12  5000.3  758.79  5010.3  773.92
  5020.3  794.48  5030.3  805.13  5040.3  807.64  5100.3  815.61  5110.3  816.47
  5120.3  817.87  5150.4  820.56  5160.4   821.8  5210.4  826.26  5219.6  826.51
#Mann= 3 ,-1 , 0
  4708.6     .12       0  4984.3     .05       0  4996.4     .12       0
Bank Sta=4984.3,4996.4
XS Rating Curve= 0 ,0
Exp/Cntr=0.3,0.1

Type RM Length L Ch R = 1 ,11391   ,192,192,192
BEGIN DESCRIPTION:
Dry Comal Creek Tributary 13 17.0
END DESCRIPTION:
XS GIS Cut Line= 3
      2217575.02     13794575.01        2217425.       13794475.
        2217325.       13794475.
#Sta/Elev= 30
  4819.3  787.27  4822.3  787.27  4841.9  786.18  4847.9  785.59  4855.4  784.46
  4868.9  781.59    4905     775    4914  771.93    4920  769.46  4927.5  767.01
    4941  766.29    4950  766.43  4963.5  763.25  4971.1  762.98  4977.1   761.9
  4986.1  761.13  4996.6  759.21  5002.1  759.21  5003.6  756.96  5004.1  756.46
  5015.2  756.46  5015.7  756.96  5029.6  763.69  5039.6  777.18  5049.6  791.59
  5059.6  812.07  5069.6  818.58  5079.6  821.84  5089.6  822.89  5099.6  823.39
#Mann= 3 ,-1 , 0
  4819.3     .12       0  5003.6     .05       0  5015.7     .12       0
Bank Sta=5003.6,5015.7
XS Rating Curve= 0 ,0
Exp/Cntr=0.3,0.1

Type RM Length L Ch R = 1 ,11199   ,255,255,255
BEGIN DESCRIPTION:
X18982
END DESCRIPTION:
XS GIS Cut Line= 2
       2217753.9     13794492.26      2217411.57     13794222.25
#Sta/Elev= 30
  4753.4  789.17    4801  787.81  4850.7  783.98  4871.5  781.25    4886  780.06
  4900.4  775.46  4906.8  772.17  4914.9  769.52  4921.2  764.97  4935.7  760.59
  4956.5  757.48  4964.6  758.36  4970.9  757.78  4993.4  755.01  4993.8  754.42
  4994.3  753.92  5005.4  753.92  5005.9  754.42  5020.6  761.05  5028.7  768.61
  5035.1  782.93  5043.1  793.05  5049.5  802.26  5057.6  806.12  5063.9  808.14
  5070.4  811.99  5092.8  817.47  5128.1  821.99  5171.4  824.27  5189.4  824.55
#Mann= 3 ,-1 , 0
  4753.4     .12       0  4993.8     .05       0  5005.9     .12       0
Bank Sta=4993.8,5005.9
XS Rating Curve= 0 ,0
Exp/Cntr=0.3,0.1

Type RM Length L Ch R = 1 ,10944   ,443,443,443
BEGIN DESCRIPTION:
Dry Comal Creek Tributary 13 16.0
END DESCRIPTION:
XS GIS Cut Line= 3
      2217874.98     13794324.98        2217775.       13794225.
      2217675.02     13794125.02
#Sta/Elev= 27
  4858.6  782.78  4862.1  782.78  4872.7  781.56  4886.9  780.26  4893.9  779.46
    4901  777.61  4915.1  772.14  4929.3   762.6  4943.4  758.22  4971.7  756.36
  4985.9  752.73  4990.4   751.4  4990.9   750.9    5002   750.9  5002.5   751.4
  5003.5   751.4  5014.1  752.32  5028.3  754.75  5042.4  763.06  5056.6  769.88
  5070.7  780.07  5084.9  793.99    5099  806.96  5113.1  811.14  5127.3  812.76
  5137.9  813.31  5141.4  813.31
#Mann= 3 ,-1 , 0
  4858.6     .12       0  4990.4     .05       0  5002.5     .12       0
Bank Sta=4990.4,5002.5
XS Rating Curve= 0 ,0
Exp/Cntr=0.3,0.1

Type RM Length L Ch R = 1 ,10501   ,266,266,266
BEGIN DESCRIPTION:
Dry Comal Creek Tributary 13 15.0
END DESCRIPTION:
XS GIS Cut Line= 3
      2218224.98     13794174.96        2218175.       13794075.
      2218025.03     13793975.02
#Sta/Elev= 30
    4883  775.94  4885.8  775.94  4891.3  774.79  4896.9  774.59  4919.3  769.89
  4927.7  765.52  4936.1  759.89  4941.7  760.08    4950  754.11  4958.4  751.35
  4980.3   750.8  4980.8   750.3  4991.9   750.3  4992.4   750.8  5023.3  752.45
  5038.3  752.44  5044.3  751.22  5074.4  754.68  5080.4  760.84  5089.4   763.5
  5095.4  770.58  5102.9  774.51  5110.4   779.1  5116.4  784.07  5125.5  786.78
  5131.5  790.15    5139   792.5  5167.5  796.27    5172  797.22    5175  797.22
#Mann= 3 ,-1 , 0
    4883     .12       0  4980.3     .05       0  4992.4     .12       0
Bank Sta=4980.3,4992.4
XS Rating Curve= 0 ,0
Exp/Cntr=0.3,0.1

Type RM Length L Ch R = 1 ,10235   ,205,205,205
BEGIN DESCRIPTION:
X18983
END DESCRIPTION:
XS GIS Cut Line= 2
      2218486.61     13794145.12      2218318.37     13793799.04
#Sta/Elev= 30
  4788.9  786.21  4827.4  783.59    4850  780.72  4855.7  778.56  4872.5  775.14
  4878.1  774.07  4895.1  772.86  4900.6  770.79  4917.6  771.16  4923.2  769.81
  4933.6  769.96  4940.2  768.89  4945.8  766.41  4955.8  764.67  4962.7  761.92
  4968.3  753.11  4978.1  742.52  4984.8     740  4985.3   739.5    4997     740
  5000.3  742.01  5007.9  742.12  5022.5  744.23  5030.4  747.27    5053  759.59
    5067  763.82  5111.5  772.75  5143.2  777.81  5148.8     780  5173.7  784.12
#Mann= 3 ,-1 , 0
  4788.9     .12       0  4984.8     .05       0    4997     .12       0
Bank Sta=4984.8,4997
XS Rating Curve= 0 ,0
Exp/Cntr=0.3,0.1

Type RM Length L Ch R = 1 ,10030   ,438,438,438
BEGIN DESCRIPTION:
Dry Comal Creek Tributary 13 14.0
END DESCRIPTION:
XS GIS Cut Line= 3
        2218625.       13793975.        2218575.       13793875.
        2218525.     13793725.01
#Sta/Elev= 30
  4883.9  780.51  4886.7  780.51  4897.9  778.82  4914.6  775.06  4920.2  775.06
  4928.6  772.96    4937  770.05  4942.6  770.36    4951  767.78    4965   760.2
  4973.3  753.99  4981.7  749.46  4987.3  748.29  4992.9  744.16  4998.3  744.16
  5006.2  738.11  5010.7  736.02  5011.2  735.52  5022.4  735.52  5022.9  736.02
  5027.3   737.8  5048.4   743.6  5058.9  745.92  5069.5  749.48    5080  757.43
  5090.6   763.2  5111.7  772.31  5122.2   774.2  5132.7  775.22  5153.8  776.17
#Mann= 3 ,-1 , 0
  4883.9     .12       0  5010.7     .05       0  5022.9     .12       0
Bank Sta=5010.7,5022.9
XS Rating Curve= 0 ,0
Exp/Cntr=0.3,0.1

Type RM Length L Ch R = 1 ,9592    ,454,454,454
BEGIN DESCRIPTION:
Dry Comal Creek Tributary 13 13.0
END DESCRIPTION:
XS GIS Cut Line= 3
      2218924.99     13793724.96        2218875.       13793575.
      2218774.98     13793524.99
#Sta/Elev= 30
  4849.3  776.01  4859.8  775.07  4870.3  775.51  4880.9  772.86  4891.4  768.96
    4902  763.49    4923  755.88  4933.6  749.53  4944.1   745.8  4954.7  743.65
  4975.8  733.12  4986.3  731.01  4990.7  729.52  4991.2  729.02  5002.4  729.02
  5002.9  729.52  5004.7  731.59  5010.2  731.59  5015.8  738.62  5021.4  739.91
  5029.7  743.21  5043.7  747.08  5060.5  751.33  5066.1  752.33  5082.8  758.73
  5088.4  759.74  5105.2  766.66  5110.8  766.81  5116.4  769.25  5119.2  769.25
#Mann= 3 ,-1 , 0
  4849.3     .12       0  4990.7     .05       0  5002.9     .12       0
Bank Sta=4990.7,5002.9
XS Rating Curve= 0 ,0
Exp/Cntr=0.3,0.1

Type RM Length L Ch R = 1 ,9138    ,426,426,426
BEGIN DESCRIPTION:
Dry Comal Creek Tributary 13 12.0
END DESCRIPTION:
XS GIS Cut Line= 3
      2219325.02     13793375.02        2219125.       13793225.
      2218975.03       13793225.
#Sta/Elev= 30
  4749.6  778.79  4799.6  773.14  4813.2  770.01  4821.5  767.15  4827.8  765.88
  4836.1   761.5  4842.3  759.53  4856.9  752.82  4871.5  748.09  4886.1   744.5
  4906.9  741.58  4927.8  734.89  4942.3  734.37  4943.5  733.84    4944  733.34
  4955.3  733.34  4955.8  733.84  4956.9  735.22  4963.2  734.42  4971.5  735.59
  5002.1  734.42  5019.6  738.78  5039.6  745.68  5049.6  747.02  5059.6  747.57
  5069.6  746.98  5079.6  749.18  5099.6  751.44  5119.6  756.41  5149.6  760.81
#Mann= 3 ,-1 , 0
  4749.6     .12       0  4943.5     .05       0  4955.8     .12       0
Bank Sta=4943.5,4955.8
XS Rating Curve= 0 ,0
Exp/Cntr=0.3,0.1

Type RM Length L Ch R = 1 ,8712    ,480,480,480
BEGIN DESCRIPTION:
Dry Comal Creek Tributary 13 11.0
END DESCRIPTION:
XS GIS Cut Line= 3
      2219725.01       13792875.        2219325.       13792875.
      2218925.01     13793024.99
#Sta/Elev= 30
  4604.6  798.01  4644.6  790.77  4654.6   787.5  4684.6     774  4714.6  762.53
  4734.6   756.5  4754.6  749.34  4764.6  746.93  4804.6  742.69  4874.6  740.78
  4924.6  738.41  4934.6  736.47  4964.6  728.61  4974.6  727.45  4978.4  726.03
  4978.9  725.53  4990.3  725.53  4990.8  726.03  4994.6   728.2  5002.1  729.05
  5019.7  728.74  5044.7  732.21    5050  731.83    5058  733.33  5074.9  734.89
  5143.5  739.35    5325  742.09  5356.2  743.62  5386.4  747.05  5431.8  749.74
#Mann= 3 ,-1 , 0
  4604.6     .12       0  4978.4     .05       0  4990.8     .12       0
Bank Sta=4978.4,4990.8
XS Rating Curve= 0 ,0
Exp/Cntr=0.3,0.1

Type RM Length L Ch R = 1 ,8232    ,456,456,456
BEGIN DESCRIPTION:
Dry Comal Creek Tributary 13 10.0
END DESCRIPTION:
XS GIS Cut Line= 3
      2219775.05     13792525.01        2219325.       13792425.
      2219125.02       13792425.
#Sta/Elev= 30
  4543.9  797.84  4584.9   795.4  4605.4  789.04  4611.8  785.58  4616.9  785.22
  4655.4  772.91  4659.2  773.15  4687.4  765.56  4697.6  760.69    4704  755.53
  4709.1  756.55  4747.5  738.66  4752.7  739.79  4759.1  735.91  4769.3   732.9
  4801.3  732.55  4839.7  734.83  4861.5  731.49  4902.5  731.02  4937.1  728.14
  4953.7  722.15  4979.2  720.04  4979.7  719.54  4992.3  720.04  4994.7  721.44
  5007.4  722.65  5034.9  733.52  5064.9  738.71  5174.9  752.43  5204.9  753.57
#Mann= 3 ,-1 , 0
  4543.9     .12       0  4979.2     .05       0  4992.3     .12       0
Bank Sta=4979.2,4992.3
XS Rating Curve= 0 ,0
Exp/Cntr=0.3,0.1

Type RM Length L Ch R = 1 ,7776    ,439,439,439
BEGIN DESCRIPTION:
Dry Comal Creek Tributary 13 9.0
END DESCRIPTION:
XS GIS Cut Line= 3
      2219575.02       13792075.        2219375.       13792025.
      2219024.99       13791775.
#Sta/Elev= 30
    4782  757.54    4916  747.36  4928.9  744.73  4957.3  730.23    4965  724.36
  4970.1  724.74  4985.6  720.62  4995.5   720.6  5009.8     716  5010.3   715.5
    5023     716    5025  720.56  5037.3  717.55  5060.7  719.12  5102.5   718.4
  5123.4  725.65    5132  726.45  5173.7  724.38  5238.9  726.18  5253.6  734.17
  5259.8  733.75  5268.4  743.98  5274.5  742.59  5283.1  755.34    5304  766.49
  5324.9  773.68  5339.6  783.07  5369.1  795.13  5404.8  803.76  5418.3   804.8
#Mann= 3 ,-1 , 0
    4782     .12       0  5009.8     .05       0    5023     .12       0
Bank Sta=5009.8,5023
XS Rating Curve= 0 ,0
Exp/Cntr=0.3,0.1

Type RM Length L Ch R = 1 ,7337    ,458,458,458
BEGIN DESCRIPTION:
Dry Comal Creek Tributary 13 8.0
END DESCRIPTION:
XS GIS Cut Line= 3
      2219524.98     13791874.98        2219325.       13791625.
      2219174.97     13791474.97
#Sta/Elev= 30
  4679.8   747.5  4715.8  744.48    4751  739.28  4757.4   737.4  4765.4  736.79
  4786.2  732.55  4821.4  727.58  4871.9  723.77  4885.5  721.57  4907.9  721.43
  4914.3  719.97  4922.3  719.67  4928.7  717.51  4943.1  715.28  4957.5  714.31
  4963.9  712.21  4971.9  710.98  4990.1  709.18  4990.6  708.68  5003.3  709.18
  5014.1  709.49  5028.2  725.55  5035.3  727.11  5042.4  737.34  5056.5  749.74
  5070.6  759.99  5113.1  771.18  5183.8  793.16  5197.9   796.7  5212.1  798.57
#Mann= 3 ,-1 , 0
  4679.8     .12       0  4990.1     .05       0  5003.3     .12       0
Bank Sta=4990.1,5003.3
XS Rating Curve= 0 ,0
Exp/Cntr=0.3,0.1

Type RM Length L Ch R = 1 ,6879    ,477,477,477
BEGIN DESCRIPTION:
Dry Comal Creek Tributary 13 7.0
END DESCRIPTION:
XS GIS Cut Line= 3
        2219675.     13791774.98        2219675.       13791425.
      2219525.01     13791275.01
#Sta/Elev= 30
    4650   747.7    4690  746.54    4700  740.58    4720  742.45    4730  744.36
    4740  741.11    4750  739.68    4760  736.72    4770  731.59    4780  729.54
    4810  725.92    4850  717.96    4870  715.82    4890   716.7    4910  715.67
    4950  710.48    4990  702.57  5014.1  702.51  5021.7  701.57  5022.2  701.07
  5034.9  701.57  5042.4  713.11  5056.5  736.68  5070.7  746.42  5084.8  753.16
    5099  758.09  5127.3  766.03  5141.4  767.28  5169.7  771.42  5212.1  774.12
#Mann= 3 ,-1 , 0
    4650     .12       0  5021.7     .05       0  5034.9     .12       0
Bank Sta=5021.7,5034.9
XS Rating Curve= 0 ,0
Exp/Cntr=0.3,0.1

Type RM Length L Ch R = 1 ,6402    ,456,456,456
BEGIN DESCRIPTION:
Dry Comal Creek Tributary 13 6.0
END DESCRIPTION:
XS GIS Cut Line= 3
      2220024.99     13791825.03        2220125.       13791525.
      2220024.98     13791324.97
#Sta/Elev= 30
    4676  751.83  4686.6  751.04  4760.4   734.3  4781.4  731.71  4823.6  720.55
  4855.2  714.34  4886.9  710.44  4907.9  709.96  4939.6  704.66  4950.1  699.76
    4966  699.41  4999.6  698.84  5000.1  698.34  5012.8  698.84    5037  703.48
  5041.3  711.82  5045.4  719.77    5051  713.79  5059.3   724.5  5067.7  729.61
  5073.3  727.87  5081.7  735.62  5090.1  741.15  5095.7  740.72    5118  744.99
  5134.8   750.8  5157.2  756.22  5171.1  758.07  5205.3  758.55  5215.9  758.77
#Mann= 6 ,-1 , 0
    4676     .12       0    4966    .035       0  4999.6    .035       0
  5012.8    .035       0  5041.3     .12       0  5205.3    .035       0
Bank Sta=4999.6,5012.8
XS Rating Curve= 0 ,0
Exp/Cntr=0.3,0.1

Type RM Length L Ch R = 1 ,5946    ,202,202,202
BEGIN DESCRIPTION:
Dry Comal Creek Tributary 13 5.0
END DESCRIPTION:
XS GIS Cut Line= 3
        2220575.     13791874.99        2220525.       13791675.
        2220325.       13791375.
#Sta/Elev= 30
  4789.7  765.17  4854.1  753.33  4882.5  743.76  4895.3  740.63  4923.7  739.53
  4936.6  734.81  4944.3  729.16  4964.9  720.87  4985.5  707.34  4993.3   694.9
  4995.8   694.9  4996.6  689.23  4997.1  688.73  5010.2  689.23  5031.9   691.2
  5039.4   693.8  5060.4  695.55    5068  697.45  5081.5  697.38  5111.5  700.41
  5168.6  703.08  5183.6  706.93  5204.7  709.06  5219.7  713.31  5240.7  717.11
  5248.2  720.26  5270.8  723.61  5312.8  733.46  5327.9  736.06  5356.4  737.35
#Mann= 3 ,-1 , 0
  4789.7     .12       0  4996.6     .05       0  5010.2     .12       0
Bank Sta=4996.6,5010.2
XS Rating Curve= 0 ,0
Exp/Cntr=0.3,0.1

Type RM Length L Ch R = 1 ,5744    ,254,254,254
BEGIN DESCRIPTION:
X18980
END DESCRIPTION:
XS GIS Cut Line= 2
      2220872.84     13791778.15      2220376.35     13791315.41
#Sta/Elev= 30
    4775   783.3  4832.3  780.49  4888.9  774.88  4917.3  760.02  4924.1  753.45
  4938.3  737.06  4945.6  730.68  4952.4  721.06  4959.8  715.36  4966.6     707
  4973.9  702.79  4980.8  695.99  4988.1  694.62  4994.9  691.62  5002.3  691.19
  5009.6  687.44  5010.1  686.94  5023.2  687.44  5023.3  688.47  5030.6  687.82
  5051.6  690.41  5065.8  695.16  5086.8  698.44  5129.3  701.42  5179.1  702.71
  5285.1  715.29  5299.3  718.88    5377  730.31  5426.8  736.04  5453.7   737.5
#Mann= 3 ,-1 , 0
    4775     .12       0  5009.6     .05       0  5023.2     .12       0
Bank Sta=5009.6,5023.2
XS Rating Curve= 0 ,0
Exp/Cntr=0.3,0.1
