--- GERONIMO CREEK.prj (project) ---

Proj Title=GERONIMO CREEK Base Level Engineering
Current Plan=p01
Default Exp/Contr=0.3,0.1
English Units
Geom File=g01
Flow File=f01
Plan File=p01
Y Axis Title=Elevation
X Axis Title(PF)=Main Channel Distance
X Axis Title(XS)=Station
BEGIN DESCRIPTION:
GERONIMO CREEK
END DESCRIPTION:
DSS Export Rating Curves= 0
DSS Export Rating Curve Sorted= 0
DSS Export Volume Flow Curves= 0
DXF OffsetX= 0
DXF OffsetY= 0
DXF ScaleX= 1
DXF ScaleY= 10

--- GERONIMO CREEK.p01 (plan) ---

Plan Title=Multiple Run
Program Version=4.10
Short Identifier=Multiple
Geom File=g01
Flow File=f01
Subcritical Flow
K Sum by GR= 0
Std Step Tol= 0.01
Critical Tol= 0.01
Num of Std Step Trials= 20
Max Error Tol= 0.3
Flow Tol Ratio= 0.001
Split Flow NTrial= 30
Split Flow Tol= 0.02
Split Flow Ratio= 0.02
Log Output Level= 0
Friction Slope Method= 1
Unsteady Friction Slope Method= 2
Unsteady Bridges Friction Slope Method= 1
Parabolic Critical Depth
Global Vel Dist= 1 , 1 , 1
Global Log Level= 0
CheckData=True
Encroach Param=-1 ,0,0, 0
BEGIN DESCRIPTION:
Multiple Run
END DESCRIPTION:
Computation Interval=1HOUR
Output Interval=1HOUR
Run HTab= 0
Run UNet= 0
Run PostProcess= 0
Run WQNet= 0
UNET Theta= 1
UNET Theta Warmup= 1
UNET ZTol= 0.02
UNET ZSATol= 0.05
UNET MxIter= 20
UNET MaxInSteps= 0
UNET DtIC= 0
UNET DtMin= 0
UNET MaxCRTS= 20
UNET WFStab= 2
UNET SFStab= 1
UNET WFX= 1
UNET SFX= 1
UNET DSS MLevel= 4
UNET DZMax Abort= 100
UNET Convert EG Bridges= 0
UNET Use Existing IB Tables=-1
UNET Froude Reduction=False
UNET Froude Limit= 1
UNET Froude Power= 10
UNET Time Slicing=0,0, 5
UNET Junction Losses=0
Instantaneous Interval=1HOUR
Write IC File= 0
Write IC File at Sim End=0
Echo Input=False
Echo Parameters=False
Echo Output=False
Write Detailed= 0
WQ AD Non Conservative
WQ ULTIMATE=-1
WQ Max Comp Step=1HOUR
WQ Output Interval=15MIN
WQ Output Selected Increments= 0
WQ Output face flow=0
WQ Output face velocity=0
WQ Output face area=0
WQ Output face dispersion=0
WQ Output cell volume=0
WQ Output cell surface area=0
WQ Output cell continuity=0
WQ Output cumulative cell continuity=0
WQ Output face conc=0
WQ Output face dconc_dx=0
WQ Output face courant=0
WQ Output face peclet=0
WQ Output face adv mass=0
WQ Output face disp mass=0
WQ Output cell mass=0
WQ Output cell source sink temp=0
WQ Output cell source sink nsm=0
WQ Output MaxMinRange=-1
WQ Daily Max Min Mean=-1
WQ Daily Range=0
WQ Daily Time=0
WQ Create Restart=0
WQ Fixed Restart=0
WQ System Summary=0
WQ Use Fixed Temperature=0
Sorting and Armoring Iterations= 10
XS Update Threshold= 0.02
Hydraulics Update Threshold= 0.02
Energy Slope Method= 1
Volume Change Method= 0
XS Weighting Method= 0
Number of US Weighted Cross Sections= 1
Number of DS Weighted Cross Sections= 1
Upstream XS Weight=0.25
Main XS Weight=0.5
Downstream XS Weight=0.25
Number of DS XS's Weighted with US Boundary= 1
Upstream Boundary Weight= 1
Weight of XSs Associated with US Boundary= 0
Number of US XS's Weighted with DS Boundary= 1
Downstream Boundary Weight= 0.5
Weight of XSs Associated with DS Boundary= 0.5
Sediment Output Level= 4
Mass or Volume Output= 0
Output Increment Type= 1
Profile and TS Output Increment= 10
XS Output Flag= 0
XS Output Increment= 10
Disregard all LS=0
Disregard all Conn=0
Disregard all Breaches=0
Disregard all Pumps=0

--- GERONIMO CREEK.f01 (steady flow) ---

Flow Title=Multiple
Program Version=4.10
Number of Profiles= 7
Profile Names=10-year,25-year,50-year,1pct_min,100-year,1pct_plu,500-year
River Rch & RM=GERONIMO CREEK,Reach-1         ,97935
     465     714     926     580    1157    2309    1789
River Rch & RM=GERONIMO CREEK,Reach-1         ,96269
     927    1497    2009    1301    2596    5180    4294
River Rch & RM=GERONIMO CREEK,Reach-1         ,95403
    1070    1727    2318    1500    2992    5970    4938
River Rch & RM=GERONIMO CREEK,Reach-1         ,89475
    1353    2213    2996    1954    3899    7780    6543
River Rch & RM=GERONIMO CREEK,Reach-1         ,85334
    1417    2326    3157    2066    4122    8224    6966
River Rch & RM=GERONIMO CREEK,Reach-1         ,79215
    5106    8816   12386    8364   16688   33297   30029
River Rch & RM=GERONIMO CREEK,Reach-1         ,74277
    5388    9315   13101    8855   17668   35252   31849
River Rch & RM=GERONIMO CREEK,Reach-1         ,70128
    5373    9275   13030    8796   17550   35017   31559
River Rch & RM=GERONIMO CREEK,Reach-1         ,65828
    5579    9644   13560    9161   18279   36472   32926
River Rch & RM=GERONIMO CREEK,Reach-1         ,64898
    6118   10597   14922   10095   20142   40189   36373
River Rch & RM=GERONIMO CREEK,Reach-1         ,61758
    6004   10423   14697    9955   19862   39631   35972
River Rch & RM=GERONIMO CREEK,Reach-1         ,60638
    6030   10465   14755    9993   19939   39783   36100
River Rch & RM=GERONIMO CREEK,Reach-1         ,57894
    6121   10626   14984   10150   20252   40408   36678
River Rch & RM=GERONIMO CREEK,Reach-1         ,55750
    6213   10790   15218   10309   20570   41043   37264
River Rch & RM=GERONIMO CREEK,Reach-1         ,50742
    6178   10720   15110   10230   20412   40727   36932
River Rch & RM=GERONIMO CREEK,Reach-1         ,47404
    6781   11794   16654   11294   22534   44961   40897
River Rch & RM=GERONIMO CREEK,Reach-1         ,46190
    6873   11962   16899   11464   22874   45640   41550
River Rch & RM=GERONIMO CREEK,Reach-1         ,43511
    6878   11958   16880   11443   22831   45554   41404
River Rch & RM=GERONIMO CREEK,Reach-1         ,38591
    6880   11958   16877   11438   22822   45535   41370
River Rch & RM=GERONIMO CREEK,Reach-1         ,37641
    7646   13319   18828   12779   25498   50875   46350
River Rch & RM=GERONIMO CREEK,Reach-1         ,30849
    7657   13340   18858   12801   25540   50960   46433
River Rch & RM=GERONIMO CREEK,Reach-1         ,30423
    7871   13727   19421   13192   26322   52520   47925
River Rch & RM=GERONIMO CREEK,Reach-1         ,26645
    8140   14211   20120   13676   27287   54446   49746
River Rch & RM=GERONIMO CREEK,Reach-1         ,17837
    8166   14248   20165   13701   27338   54546   49795
River Rch & RM=GERONIMO CREEK,Reach-1         ,15340
    8436   14714   20820   14141   28216   56298   51360
River Rch & RM=GERONIMO CREEK,Reach-1         ,10028
    8474   14775   20902   14195   28322   56509   51530
River Rch & RM=GERONIMO CREEK,Reach-1         ,5771
    8636   15076   21345   14508   28946   57756   52755
Boundary for River Rch & Prof#=GERONIMO CREEK,Reach-1         , 1
Up Type= 0
Dn Type= 3
Dn Slope=0.0008
Boundary for River Rch & Prof#=GERONIMO CREEK,Reach-1         , 2
Up Type= 0
Dn Type= 3
Dn Slope=0.0008
Boundary for River Rch & Prof#=GERONIMO CREEK,Reach-1         , 3
Up Type= 0
Dn Type= 3
Dn Slope=0.0008
Boundary for River Rch & Prof#=GERONIMO CREEK,Reach-1         , 4
Up Type= 0
Dn Type= 3
Dn Slope=0.0008
Boundary for River Rch & Prof#=GERONIMO CREEK,Reach-1         , 5
Up Type= 0
Dn Type= 3
Dn Slope=0.0008
Boundary for River Rch & Prof#=GERONIMO CREEK,Reach-1         , 6
Up Type= 0
Dn Type= 3
Dn Slope=0.0008
Boundary for River Rch & Prof#=GERONIMO CREEK,Reach-1         , 7
Up Type= 0
Dn Type= 3
Dn Slope=0.0008
DSS Import GetInterval= 0
DSS Import GetPeak= 0
DSS Import FillOption= 0

--- GERONIMO CREEK.g01 (geometry) ---

Geom Title=Existing Conditions
Program Version=4.10

River Reach=GERONIMO CREEK  ,Reach-1
Reach XY= 30
        2275875.       13798725.      2276869.07     13799522.76
      2281077.67     13797369.58      2284868.95     13793483.16
      2287630.86     13792677.06      2289799.63      13793325.4
       2293264.5      13792776.2      2295523.54     13794271.47
      2297580.18     13790330.41      2300517.25     13789681.19
      2302323.81      13786714.5      2301384.03     13785167.99
      2302415.32     13783285.78      2303914.37       13783135.
      2304823.39     13780818.98      2303674.66     13780000.22
      2305123.72     13778218.96      2304678.61      13775926.5
      2307291.76     13774908.57      2308472.85     13772419.03
      2308621.25     13769776.55        2305675.       13767275.
        2305425.       13764375.      2306971.46     13764023.54
      2306024.96     13762859.66      2306528.45     13760576.25
      2310321.24     13756423.44      2311367.44       13753675.
      2311227.26     13749430.94        2313625.       13745875.

Type RM Length L Ch R = 1 ,97935   ,593,593,593
BEGIN DESCRIPTION:
A18964
END DESCRIPTION:
XS GIS Cut Line= 3
      2274678.73      13799703.3      2275946.93     13798725.86
      2276299.56     13797395.77
#Sta/Elev= 30
  3449.5  634.09  3895.1  632.01  4265.4  629.49  4351.7  629.69    4358  629.27
  4366.2  629.71  4372.5  629.28  4401.5  630.25  4407.8  629.74    4416  630.15
  4422.3  629.75    4493  630.14  4586.3  629.93  4600.8  629.45  4607.1  629.91
  4615.3  629.43  4636.1  629.79  4650.6   629.2  4957.8  628.63  4997.3  626.75
  4997.6  626.25  5001.2  626.25  5001.5  626.75  5047.3  628.27  5248.1  629.71
  5687.4  630.81  5880.2  631.92  5930.9  632.48  6054.3  632.58  6426.7  633.41
#Mann= 5 ,-1 , 0
  3449.5    .045       0  4997.3    .045       0  5001.5    .045       0
  5880.2    .035       0  6054.3    .045       0
Bank Sta=4997.3,5001.5
XS Rating Curve= 0 ,0
Exp/Cntr=0.3,0.1

Type RM Length L Ch R = 1 ,97342   ,618,618,618
BEGIN DESCRIPTION:
A18963
END DESCRIPTION:
XS GIS Cut Line= 3
      2274907.67     13800130.12      2276256.25     13799202.21
      2276750.57     13797725.41
#Sta/Elev= 30
    3438  633.84  3699.3  633.26  4057.8  630.81  4374.4  629.63  4583.4  627.59
  5005.4  625.72  5005.6  625.22  5009.3  625.22  5009.6  625.72    5182  626.78
  5356.7  629.51    5536  630.57  5599.3  630.82  6007.3  630.13  6073.8  630.07
  6092.3  630.69    6116  630.13  6155.4  630.96  6160.7  630.62  6185.3  630.81
  6218.6  630.92  6223.8  630.53  6281.7  631.12    6287  630.76  6344.9  631.22
  6350.1  630.73  6376.4  631.12  6381.7  630.77    6408  631.14  6632.3  631.39
#Mann= 5 ,-1 , 0
    3438    .045       0  5005.4    .045       0  5009.6    .045       0
  6007.3    .035       0  6185.3    .045       0
Bank Sta=5005.4,5009.6
XS Rating Curve= 0 ,0
Exp/Cntr=0.3,0.1

Type RM Length L Ch R = 1 ,96724   ,455,455,455
BEGIN DESCRIPTION:
GERONIMO CREEK 31.0
END DESCRIPTION:
XS GIS Cut Line= 3
      2275475.01     13801324.98        2276675.       13799525.
      2276819.04     13797738.01
#Sta/Elev= 30
  2836.7  633.14  3571.3  629.98  3724.5  628.48  3774.1  627.26  3846.2  628.46
  4178.2  627.83  4278.9  627.26  4394.6  627.96    4964  624.54  5160.5  625.06
  5306.4  624.42  5306.7  623.92  5310.4  623.92  5310.7  624.42  5381.2  624.84
    5436  625.74  5531.7  629.22  5591.9  630.12  5642.1  630.41  5832.7  629.73
  6005.8  629.81  6073.5  629.61  6083.5  629.13  6103.6  629.32  6133.7   628.6
  6180.6  630.39  6185.6     630  6219.8  630.59  6334.3  629.34  6792.8  630.96
#Mann= 5 ,-1 , 0
  2836.7    .045       0  5306.4    .045       0  5310.7    .045       0
  6005.8    .035       0  6219.8    .045       0
Bank Sta=5306.4,5310.7
XS Rating Curve= 0 ,0
Exp/Cntr=0.3,0.1

Type RM Length L Ch R = 1 ,96269   ,424,424,424
BEGIN DESCRIPTION:
GERONIMO CREEK 30.0
END DESCRIPTION:
XS GIS Cut Line= 3
      2276474.99     13801375.04        2277075.       13799375.
      2276856.32     13797785.57
#Sta/Elev= 30
  2912.4  631.56  3340.5  630.01  3698.1  627.74  3764.2  626.89  3998.2  626.71
  4039.1     626  4044.3  626.35  4060.9   625.4  4352.3  625.82  4729.1  624.98
  4987.9  623.49  4988.2  622.99    4992  622.99  4992.3  623.49  5283.1  624.05
  5495.1  626.34  5623.7  626.84  5694.7  626.75  5727.3  627.33  5766.7  626.57
  5771.8  627.11  5787.8  626.25  5828.2  627.57  5900.3  628.81  5979.6  627.87
  6110.9  628.91  6302.7     629  6423.8  630.26  6474.3  629.62  6604.9  630.49
#Mann= 5 ,-1 , 0
  2912.4    .045       0  4987.9    .045       0  4992.3    .045       0
  5623.7    .035       0  5900.3    .045       0
Bank Sta=4987.9,4992.3
XS Rating Curve= 0 ,0
Exp/Cntr=0.3,0.1

Type RM Length L Ch R = 1 ,95845   ,442,442,442
BEGIN DESCRIPTION:
GERONIMO CREEK 29.0
END DESCRIPTION:
XS GIS Cut Line= 3
      2278174.99     13801124.98        2277375.       13799125.
      2276949.55     13797811.64
#Sta/Elev= 30
    2846  631.56  3632.2  629.31  3955.3  627.85  4515.4  624.43  4559.8  623.32
  4601.5  624.37    4966  623.31  5094.7  623.02    5144  623.19  5149.3  623.59
  5157.7  623.31    5176  621.62  5181.3  622.16  5205.8  621.07  5206.1  620.57
  5209.9  620.57  5210.2  621.07    5272   624.1    5304  624.29  5309.2  623.68
  5353.4  623.76  5629.1  626.12  5666.4   627.1  5714.8  626.29  5826.4  626.76
  5954.3  627.67  6030.2  628.97  6087.5  628.42  6151.5  629.28  6380.6  630.64
#Mann= 5 ,-1 , 0
    2846    .045       0    4966    .035       0  5205.8    .035       0
  5210.2    .035       0  5353.4    .045       0
Bank Sta=5205.8,5210.2
XS Rating Curve= 0 ,0
Exp/Cntr=0.3,0.1

Type RM Length L Ch R = 1 ,95403   ,470,470,470
BEGIN DESCRIPTION:
GERONIMO CREEK 28.0
END DESCRIPTION:
XS GIS Cut Line= 3
      2278075.01     13800625.04        2277675.       13798825.
      2276992.42     13797742.25
#Sta/Elev= 30
  3160.7  629.94    3632   628.2  4187.2  624.97  4318.3  624.71    4335  623.86
  4340.1  624.22    4349  623.68    4390  623.07  4467.5  623.22    4810  620.75
  4893.3  621.16  4998.7  619.59  4999.2  619.09    5005  619.09  5005.5  619.59
  5054.7  621.17    5070     621  5185.3  622.51  5229.3  623.58  5477.2  625.63
  5534.9  625.29  5577.3  626.17  5759.7  628.15  5802.1  627.62  5853.9  628.55
  5984.5  629.18  6042.2  629.93  6078.7  629.23  6127.7  629.98  6284.6  630.56
#Mann= 5 ,-1 , 0
  3160.7    .045       0  4187.2    .035       0  4467.5    .045       0
  4998.7    .045       0  5005.5    .045       0
Bank Sta=4998.7,5005.5
XS Rating Curve= 0 ,0
Exp/Cntr=0.3,0.1

Type RM Length L Ch R = 1 ,94933   ,468,468,468
BEGIN DESCRIPTION:
GERONIMO CREEK 27.0
END DESCRIPTION:
XS GIS Cut Line= 3
        2278075.     13800425.02        2278075.       13798625.
      2276968.86     13797638.14
#Sta/Elev= 30
  3195.2  629.33  3495.2  628.08  3773.7  626.28  3875.2  626.05  3993.3  625.19
  4195.2  624.36  4805.2  620.57  4915.2  620.67  4935.2  620.53  4985.2  619.27
    5013  619.17  5013.5  618.67  5019.5  618.67    5020  619.17  5108.5  621.07
    5300  622.65  5420.3  624.28  5667.8   626.1  5745.7  627.17  5767.3  626.62
  5979.7  629.16  6008.1  628.62  6050.7  629.36  6163.6  629.77  6213.7  630.38
  6241.5  629.73  6305.7  630.39  6404.4  630.62  6454.5  631.26  6477.6  630.52
#Mann= 5 ,-1 , 0
  3195.2    .045       0  3773.7    .035       0  3993.3    .045       0
    5013    .045       0    5020    .045       0
Bank Sta=5013,5020
XS Rating Curve= 0 ,0
Exp/Cntr=0.3,0.1

Type RM Length L Ch R = 1 ,94465   ,445,445,445
BEGIN DESCRIPTION:
GERONIMO CREEK 26.0
END DESCRIPTION:
XS GIS Cut Line= 3
        2278475.     13800224.96        2278475.       13798425.
      2276674.98     13797424.99
#Sta/Elev= 30
  3200.7  628.46  3407.2  627.54  3950.7  625.23  4420.7  622.18  4640.7  621.44
  4987.1  619.24  4987.6  618.74  4993.7  618.74  4994.2  619.24  5236.3  620.61
    5480  622.64  5588.7  624.24  6000.5  628.05  6065.7  627.88    6076   628.4
  6236.1  629.96  6271.6  629.32  6303.6  629.91  6464.9  630.67  6487.8  630.11
  6531.3  630.65  6618.2  630.73  6683.4  631.53  6715.5  630.74  6758.9  631.41
  6853.9  631.73  6899.6  632.51  6927.1  631.63  6992.3  632.44  7059.8  632.52
#Mann= 4 ,-1 , 0
  3200.7    .035       0  3407.2    .045       0  4987.1    .045       0
  4994.2    .045       0
Bank Sta=4987.1,4994.2
XS Rating Curve= 0 ,0
Exp/Cntr=0.3,0.1

Type RM Length L Ch R = 1 ,94020   ,446,446,446
BEGIN DESCRIPTION:
GERONIMO CREEK 25.0
END DESCRIPTION:
XS GIS Cut Line= 3
        2278975.       13799925.        2278775.       13798125.
      2276975.04     13797325.02
#Sta/Elev= 30
  3189.2   627.1  4004.2  624.48  4538.3  621.37  4829.2  619.67  4929.8   619.5
  4994.2  618.52  4994.7  618.02  5000.9  618.02  5001.4  618.52  5037.9  619.35
  5110.6  619.35  5255.3  620.56  5496.9   622.8  5711.6  625.35  5779.3   626.5
  5864.8  626.65  5963.3  627.96    6204  630.26  6225.9  629.52  6258.7  630.17
  6416.7  631.13    6440  630.39  6538.5     631  6590.5   630.9  6630.8  631.39
  6660.2  630.77  6849.7  632.04  6880.4  631.31  6909.2  631.87    6970  632.09
#Mann= 7 ,-1 , 0
  3189.2    .045       0  4538.3    .035       0  4994.2    .035       0
  5001.4    .035       0  5110.6    .045       0  5255.3    .035       0
  5496.9    .045       0
Bank Sta=4994.2,5001.4
XS Rating Curve= 0 ,0
Exp/Cntr=0.3,0.1

Type RM Length L Ch R = 1 ,93574   ,481,481,481
BEGIN DESCRIPTION:
GERONIMO CREEK 24.0
END DESCRIPTION:
XS GIS Cut Line= 3
        2279125.     13799675.03        2279125.       13797875.
        2277525.       13797025.
#Sta/Elev= 30
  3204.7   626.2  4094.7  623.93  4154.7  623.44  4234.7  623.47  4309.5  622.76
  4334.7  622.41  4424.7  623.11  4454.7  623.04  4592.5  620.98  4684.7  619.63
  4820.2  618.47  4924.7  618.01  4944.7  616.79  4981.1  616.12  4981.6  615.62
  4987.9  615.62  4988.4  616.12  5046.5  617.79  5072.7  618.25  5115.1  618.39
  5166.8  619.08    5435  620.96  5737.6  624.64  6024.1  627.39  6363.7  630.08
  6386.2  629.77  6431.5  630.14  6445.7  629.96  6572.2  630.81  6816.5  631.16
#Mann= 10 ,-1 , 0
  3204.7    .045       0  4309.5    .035       0  4592.5    .045       0
  4820.2    .035       0  4981.1    .035       0  4988.4    .035       0
  5046.5    .045       0  5115.1    .035       0  6024.1     .07       0
  6445.7    .045       0
Bank Sta=4981.1,4988.4
XS Rating Curve= 0 ,0
Exp/Cntr=0.3,0.1

Type RM Length L Ch R = 1 ,93093   ,447,447,447
BEGIN DESCRIPTION:
GERONIMO CREEK 23.0
END DESCRIPTION:
XS GIS Cut Line= 3
        2279175.     13799575.02        2279575.       13797775.
      2278425.02     13796175.03
#Sta/Elev= 30
  3151.8  625.88  4034.5   623.9  4134.6   623.5  4559.1  620.55  4708.9  618.73
  4738.4  617.99    4787  618.23  4792.1  617.91  4811.3  618.24  4913.8  617.04
  4954.8  617.16  4970.9  616.86  4998.8  616.47  5003.1  615.36  5034.8  615.28
  5035.3  614.78    5042  614.78  5042.5  615.28  5053.4  616.55  5081.9  617.49
  5196.4  618.22  5326.2  618.95    5504  619.86  5877.2  623.73  6042.5  625.02
  6292.2  626.68  6557.8  627.91  6655.5  628.49  6708.2  628.79  6966.1  630.26
#Mann= 11 ,-1 , 0
  3151.8    .045       0  4034.5    .035       0  4134.6    .045       0
  4970.9    .035       0  5034.8    .035       0  5042.5    .035       0
  5196.4    .045       0  5326.2    .035       0  6557.8     .07       0
  6655.5    .035       0  6708.2    .045       0
Bank Sta=5034.8,5042.5
XS Rating Curve= 0 ,0
Exp/Cntr=0.3,0.1

Type RM Length L Ch R = 1 ,92646   ,487,487,487
BEGIN DESCRIPTION:
GERONIMO CREEK 22.0
END DESCRIPTION:
XS GIS Cut Line= 3
        2279375.     13799424.99        2279975.       13797625.
      2278824.98     13796024.97
#Sta/Elev= 30
    3109  625.52  3646.1  624.14  3748.8  623.89  4352.8  620.89  4680.1  618.03
  4751.9  617.26  4890.4  614.93  4991.9  614.41  4992.4  613.91  4999.3  613.91
  4999.8  614.41  5009.4  614.45  5014.6  615.33  5070.2  615.56  5092.6  616.49
  5224.1  617.28  5314.2  617.79  5336.6  618.57  5499.9  620.43  5508.5  621.27
  5514.6  620.68  5529.3  620.41    5541  620.71  5665.6   622.3  5927.8   624.4
  6116.2  625.56  6710.1  627.89  6721.4  627.94  6866.7   629.2  6976.8  629.69
#Mann= 14 ,-1 , 0
    3109    .045       0  3646.1    .035       0  3748.8    .045       0
  4680.1    .035       0  4751.9    .045       0  4991.9    .045       0
  4999.8    .045       0  5014.6    .035       0  5224.1    .045       0
    5541    .035       0  5927.8     .07       0  6710.1    .035       0
  6721.4     .07       0  6866.7    .045       0
Bank Sta=4991.9,4999.8
XS Rating Curve= 0 ,0
Exp/Cntr=0.3,0.1

Type RM Length L Ch R = 1 ,92159   ,435,435,435
BEGIN DESCRIPTION:
GERONIMO CREEK 21.0
END DESCRIPTION:
XS GIS Cut Line= 3
      2279624.99     13799325.02        2280425.       13797525.
      2278974.98     13795924.98
#Sta/Elev= 30
  3030.2  624.98  3257.4  624.22  3363.7  623.98    3827  622.46  4288.7   620.1
  4742.1  616.27  4863.9  614.62  4956.2  614.56  4962.4  613.77  4987.1  613.73
  4987.6  613.23  4994.6  613.23  4995.1  613.73    5028  613.74  5056.4     615
  5120.6  615.13  5365.2  618.37  5566.7  620.48  5587.6  622.58  5622.8  622.13
  5686.1  622.49  5752.8  622.55    5931  623.57  6153.3  624.68  6174.6  624.75
  6295.4  625.15  6311.1  625.26  6713.6  626.74  7003.5  628.22  7159.3  629.58
#Mann= 13 ,-1 , 0
  3030.2    .045       0  3257.4    .035       0  3363.7    .045       0
  4987.1    .045       0  4995.1    .045       0  5365.2    .035       0
  5686.1    .045       0  5752.8    .035       0    5931    .045       0
  6153.3     .07       0  6174.6    .045       0  6295.4    .035       0
  6311.1    .045       0
Bank Sta=4987.1,4995.1
XS Rating Curve= 0 ,0
Exp/Cntr=0.3,0.1

Type RM Length L Ch R = 1 ,91724   ,451,451,451
BEGIN DESCRIPTION:
GERONIMO CREEK 20.0
END DESCRIPTION:
XS GIS Cut Line= 3
      2280224.99     13799225.02        2280825.       13797425.
      2279224.98     13795974.98
#Sta/Elev= 30
  3102.7  623.49  3893.3  621.46  3935.5  620.89  4135.7  620.13  4420.3  618.22
  4820.9  614.48  4926.3  613.86  4968.5  613.78    4979  614.15  4989.5  613.89
  5003.1  612.86  5003.6  612.36  5010.7  612.36  5011.2  612.86  5016.3  612.97
  5043.2   613.2    5064  613.61  5070.7  614.32  5127.5     614  5155.9  614.23
  5668.8  619.55  5673.5   619.6  5764.8  620.44  5785.7  620.94  5793.2  621.62
  5799.9  621.71  5828.3  621.45  6231.8  623.72  6677.8  625.39  7159.4  628.21
#Mann= 7 ,-1 , 0
  3102.7    .045       0  5003.1    .045       0  5011.2    .045       0
  5016.3     .07       0  5043.2    .045       0  5668.8    .035       0
  5673.5    .045       0
Bank Sta=5003.1,5011.2
XS Rating Curve= 0 ,0
Exp/Cntr=0.3,0.1

Type RM Length L Ch R = 1 ,91273   ,469,469,469
BEGIN DESCRIPTION:
GERONIMO CREEK 19.0
END DESCRIPTION:
XS GIS Cut Line= 3
      2280775.01     13799024.95        2281175.       13797225.
      2279975.01     13796025.01
#Sta/Elev= 30
  3155.9  622.29  3733.4  620.71  4058.6  619.18  4569.5  614.89  4655.3  614.68
  4917.8  612.55  4948.5  613.07    4969  612.39  4975.4  611.66  4980.6  612.12
  4997.2   610.7  5009.7  610.65  5010.2  610.15  5017.6  610.15  5018.1  610.65
    5028  611.92  5047.4  612.46    5087  613.11  5222.3  614.01  5412.1  615.01
    5622  616.42  5678.6  617.42  5763.4  617.68  5764.6  617.67  5812.9  618.06
  5876.6  617.88  5890.7  619.52  6051.1   620.4  6138.7  620.87  6696.8  624.13
#Mann= 11 ,-1 , 0
  3155.9    .045       0  5009.7    .045       0  5018.1    .045       0
  5047.4     .07       0    5087    .045       0  5222.3     .07       0
  5412.1    .045       0  5763.4    .035       0  5764.6    .045       0
  6051.1    .035       0  6138.7    .045       0
Bank Sta=5009.7,5018.1
XS Rating Curve= 0 ,0
Exp/Cntr=0.3,0.1

Type RM Length L Ch R = 1 ,90804   ,444,444,444
BEGIN DESCRIPTION:
GERONIMO CREEK 18.0
END DESCRIPTION:
XS GIS Cut Line= 3
        2281525.     13798725.02        2281525.       13796925.
      2280324.98     13795724.98
#Sta/Elev= 30
  3200.3  619.98  3770.3  619.42  4300.3  616.54  4440.3  615.15  4490.3  615.85
  4550.3  614.39  4660.3  614.08  4900.3  611.75  4950.3  612.04  4970.3  611.23
  4993.5  609.01    4994  608.51  5001.7  608.51  5002.2  609.01  5035.7  609.39
  5042.7  611.11  5056.9  612.78    5071  613.22  5141.7  611.63  5226.6  611.85
  5509.4  615.23  5636.7  615.93  5707.4  617.28  5775.8  617.53  5826.6  618.14
  5907.7  619.09  5990.3  619.67  6018.6  620.55  6240.2  621.69  6697.4  624.17
#Mann= 7 ,-1 , 0
  3200.3    .045       0  4993.5    .045       0  5002.2    .045       0
  5775.8    .035       0  5826.6    .045       0  5907.7    .035       0
  6240.2    .045       0
Bank Sta=4993.5,5002.2
XS Rating Curve= 0 ,0
Exp/Cntr=0.3,0.1

Type RM Length L Ch R = 1 ,90360   ,444,444,444
BEGIN DESCRIPTION:
GERONIMO CREEK 17.0
END DESCRIPTION:
XS GIS Cut Line= 3
        2281825.     13798424.97        2281825.       13796625.
      2280925.02     13795625.02
#Sta/Elev= 30
  3199.6  619.57  3479.6  619.48  3959.6  618.04  4459.6  615.16  4629.6  613.37
  4669.6  614.09  4709.6  612.82  4899.6  611.26  4975.2  607.94  4975.7  607.44
  4983.4  607.44  4983.9  607.94  5027.6  610.84  5063.5  611.17  5141.2  610.72
  5204.7  611.75  5275.7  611.53    5483  614.01  5608.3  616.22  5615.8  614.81
  5622.5  614.79    5630  617.28    5651  618.06  5665.2  617.89  5679.4  616.91
  5714.5  618.06  5890.3  619.53  5955.2  620.61  5997.8  620.22  6344.9  623.15
#Mann= 5 ,-1 , 0
  3199.6    .045       0  4975.2    .045       0  4983.9    .045       0
    5483    .035       0  5890.3    .045       0
Bank Sta=4975.2,4983.9
XS Rating Curve= 0 ,0
Exp/Cntr=0.3,0.1

Type RM Length L Ch R = 1 ,89916   ,441,441,441
BEGIN DESCRIPTION:
GERONIMO CREEK 16.0
END DESCRIPTION:
XS GIS Cut Line= 3
        2281975.     13798174.98        2282175.       13796375.
      2281175.01     13795475.01
#Sta/Elev= 30
  3189.3  619.37  3702.4   618.6  4165.2  616.85  4758.9  611.83  4809.2  612.67
  4849.4  611.14  4960.1  610.06  5009.8  607.64  5010.3  607.14  5018.6  607.64
  5056.8   610.4  5156.2  611.04  5276.5  609.77  5290.7   610.1  5297.5  611.51
  5304.9  611.47  5311.7  612.64  5333.3  612.99  5354.3   612.1  5375.9  612.55
  5396.9  611.54  5453.7  611.95  5482.1   612.6  5552.3  615.84  5665.9  618.36
  5955.9     621  5998.5  620.68  6062.8  621.57  6310.2  622.37  6345.7  622.86
#Mann= 5 ,-1 , 0
  3189.3    .045       0  5009.8    .045       0  5018.6    .045       0
  5156.2    .035       0  6310.2    .045       0
Bank Sta=5009.8,5018.6
XS Rating Curve= 0 ,0
Exp/Cntr=0.3,0.1

Type RM Length L Ch R = 1 ,89475   ,467,467,467
BEGIN DESCRIPTION:
GERONIMO CREEK 15.0
END DESCRIPTION:
XS GIS Cut Line= 3
        2282475.     13797874.98        2282475.       13796075.
      2281275.02     13795475.01
#Sta/Elev= 30
  3193.6  618.59  3583.6  618.68  3913.6   617.6  4333.6  614.58    4794  610.49
  4853.6  611.21  4873.6  609.57  4893.6  610.05  4920.4  609.41  4943.6  608.67
  4973.6  609.99  4983.6  608.86  4986.5  606.83    4987  606.33  4995.1  606.33
  4995.6  606.83    5002  609.04  5007.6  609.73  5029.9  610.08  5047.5  609.66
  5105.4  608.98  5264.6  609.56  5284.3  609.54  5306.6  610.45    5329  609.74
  5373.1  609.73  5449.2  610.95  5552.6  614.13  5790.2  619.46  6335.2  622.16
#Mann= 8 ,-1 , 0
  3193.6    .045       0    4794    .035       0  4920.4    .045       0
  4986.5    .045       0  4995.6    .045       0  5047.5     .07       0
  5264.6    .045       0  5373.1    .035       0
Bank Sta=4986.5,4995.6
XS Rating Curve= 0 ,0
Exp/Cntr=0.3,0.1

Type RM Length L Ch R = 1 ,89008   ,399,399,399
BEGIN DESCRIPTION:
GERONIMO CREEK 14.0
END DESCRIPTION:
XS GIS Cut Line= 3
        2282675.     13797674.99        2282875.       13795875.
      2280875.03     13795275.01
#Sta/Elev= 30
    3182  618.71    3836  617.26  4137.8  615.37  4587.7   610.8    4661  610.41
  4691.2  611.46  4751.6  608.55  4791.8  607.89  4931.6  608.52  4995.7  608.46
  5009.6   607.7  5019.8  605.87  5020.3  605.37  5028.5  605.37    5029  605.87
  5034.8  606.64  5042.7  606.28  5046.1  606.99    5087  608.41  5182.4   607.9
  5388.9   608.6  5451.5  610.04  5465.5  611.25  5556.8  610.91  5655.4  612.32
  5757.3  613.51    6125  619.58  6743.1  622.78  6757.5  623.57  7081.1  625.01
#Mann= 11 ,-1 , 0
    3182    .045       0  4587.7    .035       0  4931.6    .045       0
  5019.8    .045       0    5029    .045       0  5046.1    .035       0
  5182.4    .045       0  5451.5     .07       0  5655.4    .045       0
  5757.3    .035       0  6743.1    .045       0
Bank Sta=5019.8,5029
XS Rating Curve= 0 ,0
Exp/Cntr=0.3,0.1

Type RM Length L Ch R = 1 ,88609   ,521,521,521
BEGIN DESCRIPTION:
A18962
END DESCRIPTION:
XS GIS Cut Line= 3
      2283444.71     13797327.79      2283147.77     13795502.81
      2281724.96     13795496.62
#Sta/Elev= 30
  3274.7  617.01  3895.5  616.46  4236.5  613.59  4280.5  614.19  4334.3  612.91
  4402.1  612.42  4432.5  613.16  4469.7  611.43  4959.4  604.72  4979.6  603.67
  4985.3  602.62  4985.8  602.12  4994.7  602.62  5046.5  605.37  5127.6  606.26
  5156.4  607.87  5177.3  606.88  5195.8  606.98  5765.4  610.62  5770.4   611.6
  5776.5  611.66  5816.5  611.36  5866.5  612.18  5886.5  611.51  6025.3  613.16
  6356.5  618.18  6436.5  619.19  6466.5  618.89  6526.5  620.16  6546.5  619.82
#Mann= 8 ,-1 , 0
  3274.7    .045       0  4334.3    .035       0  4469.7    .045       0
  4985.3    .045       0  4994.7    .045       0  5177.3    .035       0
  5195.8    .045       0  6025.3    .035       0
Bank Sta=4985.3,4994.7
XS Rating Curve= 0 ,0
Exp/Cntr=0.3,0.1

Type RM Length L Ch R = 1 ,88088   ,328,328,328
BEGIN DESCRIPTION:
GERONIMO CREEK 13.0
END DESCRIPTION:
XS GIS Cut Line= 3
      2283924.99     13797074.96        2283525.       13795275.
      2281725.04       13795475.
#Sta/Elev= 30
  3151.3  616.74  3509.8  616.91  3959.2  615.11  4011.7  614.53  4032.2  614.79
  4048.9  615.84  4080.4  614.39    4369  612.69  4553.4  610.94  4922.2  606.24
  4964.4  605.48  5010.5  603.67    5011  603.17  5019.6  603.17  5020.1  603.67
  5246.7  605.79  5367.4  606.19  5387.6  606.57  5397.6  607.43  6031.5  611.06
  6041.6  611.52  6061.7  611.16  6162.3  611.85  6182.4   612.4  6222.7  612.37
  6279.5  613.59  6363.5  614.27  6665.4  618.84  6745.9  619.13  6806.2  620.21
#Mann= 6 ,-1 , 0
  3151.3    .045       0  3959.2    .035       0  4080.4    .045       0
  5010.5    .045       0  5020.1    .045       0  6279.5    .035       0
Bank Sta=5010.5,5020.1
XS Rating Curve= 0 ,0
Exp/Cntr=0.3,0.1

Type RM Length L Ch R = 1 ,87760   ,572,572,572
BEGIN DESCRIPTION:
A18961
END DESCRIPTION:
XS GIS Cut Line= 4
      2284094.27     13796393.63      2283896.31     13795131.63
      2283209.63     13794766.64      2282015.72     13794692.41
#Sta/Elev= 30
  3370.2  615.86  3475.7  615.58  3536.5  615.43  3561.1  616.44  3571.3   616.4
  3588.9  615.32  3601.6   615.1  3974.8  613.35  4298.1  610.92  5010.4  603.59
  5010.9  603.09  5019.6  603.09  5020.1  603.59  5090.8  605.12  5339.9  606.28
    5490  607.83  5512.7  608.96  5528.7  608.45  5677.6  610.48  5689.4  610.68
  5694.4  610.31  5776.2   611.5  5800.6  612.25  5874.7  612.59  6091.2  613.75
  6342.5   613.8  6461.9  613.23  6498.1  614.07    6532  613.91  6621.5  614.84
#Mann= 10 ,-1 , 0
  3370.2    .045       0  3475.7    .035       0  3536.5    .045       0
  5010.4    .045       0  5020.1    .045       0  5512.7    .035       0
  5677.6    .045       0  5776.2     .07       0  5874.7    .035       0
  6342.5    .045       0
Bank Sta=5010.4,5020.1
XS Rating Curve= 0 ,0
Exp/Cntr=0.3,0.1

Type RM Length L Ch R = 1 ,87188   ,451,451,451
BEGIN DESCRIPTION:
GERONIMO CREEK 12.0
END DESCRIPTION:
XS GIS Cut Line= 3
      2284174.99     13796374.95        2283975.       13794575.
      2282175.01       13794375.
#Sta/Elev= 30
    3189  615.88  3274.3  615.72  3329.1  615.43    3360  616.56  3410.3  615.04
  3913.4  612.87    4185  610.16    4497  608.19  4959.8  603.84  5005.2  602.76
  5005.7  602.26  5014.5  602.26    5015  602.76  5070.5  604.27  5416.6  605.51
  5459.4  605.81  5684.2   607.1  5825.1  608.86  5855.3  610.35  5945.8   610.7
  5955.9  611.26  6014.9  611.99  6113.7  613.11    6137  612.84  6331.8  614.81
  6387.8  615.26  6519.3  615.53  6549.5  616.28  6569.6  615.91  6811.1  616.64
#Mann= 11 ,-1 , 0
    3189    .045       0  3274.3    .035       0  3329.1    .045       0
  5005.2    .045       0    5015    .045       0  5416.6    .035       0
  5459.4    .045       0  6014.9    .035       0  6113.7    .045       0
  6331.8    .035       0  6387.8    .045       0
Bank Sta=5005.2,5015
XS Rating Curve= 0 ,0
Exp/Cntr=0.3,0.1

Type RM Length L Ch R = 1 ,86737   ,410,410,410
BEGIN DESCRIPTION:
GERONIMO CREEK 11.0
END DESCRIPTION:
XS GIS Cut Line= 3
      2284624.99     13796024.95        2284225.       13794225.
      2283324.98     13793024.97
#Sta/Elev= 30
  3150.9  615.42  3446.6  614.83  3949.9  612.28  4330.2  609.13  4707.9  604.81
  4737.4  605.14  4748.9  604.47  4812.6  604.16  4883.4   603.3  4921.8  603.43
  4933.3  602.86  4997.9  602.38  5002.8  601.71  5003.3  601.21  5013.3  601.21
  5013.8  601.71  5058.3  602.97  5108.7  603.25  5166.6  602.82  5316.6  603.72
  5516.6  608.45  5652.1   609.4  5857.6   612.2  5922.9  612.65  5972.9  613.69
  5987.5  613.78  5994.8  612.98  6013.9  613.24  6237.5  615.81  6494.8  617.32
#Mann= 7 ,-1 , 0
  3150.9    .045       0  4812.6    .035       0  5002.8    .035       0
  5013.8    .035       0  5108.7    .045       0  5857.6    .035       0
  6013.9    .045       0
Bank Sta=5002.8,5013.8
XS Rating Curve= 0 ,0
Exp/Cntr=0.3,0.1

Type RM Length L Ch R = 1 ,86327   ,476,476,476
BEGIN DESCRIPTION:
GERONIMO CREEK 10.0
END DESCRIPTION:
XS GIS Cut Line= 3
      2284824.99     13795674.97        2284425.       13793875.
        2284225.     13792775.02
#Sta/Elev= 30
    3165  614.48  3368.6  614.24  3779.6  612.24  4019.1  610.46  4363.5  606.32
  4382.7   606.8  4449.6  606.15  4766.7  602.88  4804.1  602.94  4892.4  603.33
  4924.7  602.68  4972.7  601.42  4973.2  600.92  4983.2  600.92  4983.7  601.42
  5029.2  602.78  5200.7  602.28  5364.6  603.24  5424.3  604.74  5435.8  604.54
  5445.9  605.75  5496.8  607.38  5506.9  609.02  5517.1  609.17  5536.1  606.84
  5557.7  608.38  5662.9  611.46  5720.2  612.02  5845.3  613.83  6126.9   616.8
#Mann= 10 ,-1 , 0
    3165    .045       0  4449.6    .035       0  4766.7    .045       0
  4804.1    .035       0  4924.7    .045       0  4972.7    .045       0
  4983.7    .045       0  5662.9    .035       0  5720.2    .045       0
  5845.3    .035       0
Bank Sta=4972.7,4983.7
XS Rating Curve= 0 ,0
Exp/Cntr=0.3,0.1

Type RM Length L Ch R = 1 ,85851   ,517,517,517
BEGIN DESCRIPTION:
GERONIMO CREEK 9.0
END DESCRIPTION:
XS GIS Cut Line= 3
        2284975.     13795375.01        2284775.       13793575.
      2284375.01     13792775.02
#Sta/Elev= 30
  3189.2  613.99  3772.8  611.17  4064.6  608.13  4084.7  609.42  4128.1   608.3
  4829.2  602.25  4927.1  602.59  4984.6  601.27  4985.1  600.77  4995.8  601.27
  5201.5  603.68  5237.9  604.76  5246.3  606.24  5260.2  606.52    5277  604.35
  5313.3   606.9  5321.7  606.98  5327.3   605.4  5344.1  609.07  5380.4  608.27
  5388.8  606.92  5402.8  608.78  5425.1  609.87  5455.9  609.37  5461.5  610.61
  5469.9  610.85  5576.9  612.36  5644.1  613.59  5688.6  614.28  5894.7  616.54
#Mann= 8 ,-1 , 0
  3189.2    .045       0  4128.1    .035       0  4927.1    .045       0
  4984.6    .045       0  4995.8    .045       0  5576.9    .035       0
  5644.1     .07       0  5688.6    .035       0
Bank Sta=4984.6,4995.8
XS Rating Curve= 0 ,0
Exp/Cntr=0.3,0.1

Type RM Length L Ch R = 1 ,85334   ,404,404,404
BEGIN DESCRIPTION:
GERONIMO CREEK 8.0
END DESCRIPTION:
XS GIS Cut Line= 4
        2285125.     13795125.05      2285213.99     13793461.33
      2285170.68     13793015.92      2284675.79      13792533.4
#Sta/Elev= 30
  3196.7  613.72    3353  613.33  3623.8  610.92  3768.1  609.69  4260.2  606.48
  4358.6  606.34    4457  604.32  4739.8   601.3  4875.3  599.31  4949.5  599.67
  4969.6   598.5  4984.1  596.35  4984.6  595.85  4995.4  596.35  4999.8  598.51
  5006.1  599.11  5170.6  601.17  5214.9  603.54  5245.2  603.03  5336.2  605.49
  5343.3  604.97  5406.9  607.58  5442.3  607.41  5470.6  608.88  5569.6  611.26
  5682.6  612.75  5739.2  614.81  5781.6  614.37  5852.4  615.92  6001.5  616.39
#Mann= 12 ,-1 , 0
  3196.7    .035       0    3353    .045       0  3623.8    .035       0
  3768.1    .045       0  4260.2    .035       0  4358.6    .045       0
    4457     .07       0  4739.8    .045       0  4875.3      .1       0
  4984.1     .05       0  4995.4      .1       0  5245.2    .035       0
Bank Sta=4984.1,4995.4
XS Rating Curve= 0 ,0
Exp/Cntr=0.3,0.1

Type RM Length L Ch R = 1 ,84930   ,449,449,449
BEGIN DESCRIPTION:
GERONIMO CREEK 7.0
END DESCRIPTION:
XS GIS Cut Line= 3
        2285175.     13794875.02        2285575.       13793325.
      2285024.98     13792674.98
#Sta/Elev= 30
  3405.2   612.4  3592.6   610.9  3733.2  609.82  4086.8  608.53  4263.4  606.64
  4338.4   606.4  4365.7  605.36  4383.4   605.9  4460.4   604.4  4655.1  601.26
  4928.9  598.01    4959  597.46  4959.5  596.96  4970.4  597.46  4983.1  598.35
  5019.7  597.86  5048.3  598.56  5148.2  597.47  5169.1  598.04  5183.4  599.96
  5204.3  600.47  5296.6  601.18  5412.2  603.31  5616.5  607.42  5651.4  609.08
  5665.7   608.5  5737.2   610.5  5765.8  610.39  5807.5     612  5857.5  612.43
#Mann= 13 ,-1 , 0
  3405.2    .045       0  3592.6    .035       0  3733.2    .045       0
  4263.4    .035       0  4338.4    .045       0  4460.4     .07       0
  4655.1    .045       0  4928.9      .1       0    4959     .05       0
  4970.4      .1       0  5148.2    .035       0  5412.2    .045       0
  5616.5    .035       0
Bank Sta=4959,4970.4
XS Rating Curve= 0 ,0
Exp/Cntr=0.3,0.1

Type RM Length L Ch R = 1 ,84481   ,439,439,439
BEGIN DESCRIPTION:
GERONIMO CREEK 6.0
END DESCRIPTION:
XS GIS Cut Line= 3
      2285424.99     13794625.03        2285975.       13793375.
      2285474.99     13792574.98
#Sta/Elev= 30
  3638.6  610.33  3660.5  610.68  3706.1  609.86  3850.7  609.66  4001.6  608.26
  4042.9  608.67  4053.8  608.04  4269.3  606.12  4512.6  603.02  4617.9  599.68
    4798  597.59  4862.3  597.83  4927.8  596.72  4937.7  595.86  4946.6  596.65
  4966.5  597.04  4995.8  595.24  4996.3  594.74  5006.7  594.74  5007.2  595.24
  5011.9  596.18  5017.8  595.56  5027.3  597.01  5033.2  596.31  5048.5  598.25
  5098.6  599.36  5106.3  600.13  5112.2  599.62  5213.6  601.01  5947.7  610.51
#Mann= 7 ,-1 , 0
  3638.6    .035       0  3706.1    .045       0    4798      .1       0
  4946.6     .07       0  4995.8     .05       0  5007.2     .07       0
  5213.6    .045       0
Bank Sta=4995.8,5007.2
XS Rating Curve= 0 ,0
Exp/Cntr=0.3,0.1

Type RM Length L Ch R = 1 ,84042   ,387,387,387
BEGIN DESCRIPTION:
GERONIMO CREEK 5.0
END DESCRIPTION:
XS GIS Cut Line= 3
      2285675.01     13794274.98        2286325.       13793475.
      2285774.99     13792674.98
#Sta/Elev= 30
  3983.3  608.64  4004.8  608.93  4021.2  607.93  4101.3  606.91  4281.4  605.04
  4495.4  601.84  4687.2  598.01  4905.1  596.35  4928.6  596.46  4957.3  595.21
  4963.8  595.57  4971.7  593.83  4978.1  593.58  4986.1   594.4  4986.7  593.27
  4987.2  592.77  4997.7  592.77  4998.2  593.27  5000.4  595.82  5006.9   594.1
  5010.8   596.1  5042.5  596.06  5057.4  594.78  5074.7  595.69  5158.9  597.97
    5219   598.5  5314.7  599.91  5340.9  600.44  5532.3  603.49  5984.9  608.18
#Mann= 10 ,-1 , 0
  3983.3    .045       0  4021.2    .035       0  4101.3    .045       0
  4905.1     .07       0  4986.7     .05       0  4998.2     .07       0
  5074.7    .045       0    5219    .035       0  5314.7     .07       0
  5340.9    .045       0
Bank Sta=4986.7,4998.2
XS Rating Curve= 0 ,0
Exp/Cntr=0.3,0.1

Type RM Length L Ch R = 1 ,83655   ,443,443,443
BEGIN DESCRIPTION:
A18960
END DESCRIPTION:
XS GIS Cut Line= 2
      2287261.63     13794420.17      2286154.32     13792434.44
#Sta/Elev= 30
  3688.3  599.67  3802.2  599.27  4079.8  596.87    4211  596.78  4490.6   597.6
  4631.8  597.28  4796.4  595.51  4908.3  594.28  4946.3  595.45  4955.2  595.45
  4967.8  594.63  4970.7  592.53  4971.2  592.03  4982.5  592.53  4983.8   593.2
  4999.5  594.64  5027.2  594.32  5056.7  596.08  5086.6  595.95  5167.8  597.43
  5189.5  596.89  5292.7  597.77  5339.3  598.18  5521.8  600.19  5531.3  600.24
  5881.1  604.21  5909.5  604.68    5922   605.8  5938.4  606.73  5961.9   606.5
#Mann= 14 ,-1 , 0
  3688.3    .035       0  3802.2     .05       0    4211     .07       0
  4490.6    .045       0  4796.4     .05       0  4946.3    .045       0
  4955.2    .035       0  4970.7    .035       0  4982.5    .035       0
  5292.7     .07       0  5339.3    .045       0  5521.8    .035       0
  5531.3    .045       0    5922     .07       0
Bank Sta=4970.7,4982.5
XS Rating Curve= 0 ,0
Exp/Cntr=0.3,0.1

Type RM Length L Ch R = 1 ,83212   ,492,492,492
BEGIN DESCRIPTION:
A18959
END DESCRIPTION:
XS GIS Cut Line= 2
       2287515.3     13794290.33      2286636.85     13792261.22
#Sta/Elev= 30
    3703  600.23  3753.4   598.6  3843.3  597.87  4033.1  597.16  4062.8  597.07
    4183  597.25  4312.2  597.96  4544.7  599.28  4743.4  598.88  4971.1  596.03
  4976.6  594.46  4999.4  593.44  4999.9  592.94  5011.7  593.44  5082.7  594.46
  5126.3  594.56  5181.3  594.76  5222.3  595.13  5266.7   596.7  5386.9  602.48
  5419.6  602.76  5478.9  605.05  5502.1  604.93  5572.2  605.91  5683.1  606.05
  5701.1  607.08  5715.6  606.68  5724.6  605.84  5840.3  606.18  5914.1  606.22
#Mann= 16 ,-1 , 0
    3703     .05       0  3753.4    .035       0  3843.3     .05       0
  4033.1     .07       0  4062.8     .05       0    4183     .07       0
  4312.2    .045       0  4999.4    .045       0  5011.7    .045       0
  5082.7     .07       0  5126.3    .035       0  5181.3     .07       0
  5266.7    .035       0  5502.1     .07       0  5715.6    .035       0
  5840.3    .045       0
Bank Sta=4999.4,5011.7
XS Rating Curve= 0 ,0
Exp/Cntr=0.3,0.1

Type RM Length L Ch R = 1 ,82720   ,454,454,454
BEGIN DESCRIPTION:
A18958
END DESCRIPTION:
XS GIS Cut Line= 2
      2287577.15     13794203.73      2287249.28     13792044.68
#Sta/Elev= 30
  3554.4  598.83  3732.7  597.31  3737.7  597.78  3795.9  596.75  3945.9  598.01
  4149.9  599.62  4170.1  598.91  4272.2  599.19  4536.9  598.02  4798.3  595.21
  4878.1  594.11  4888.2  594.72  4979.3  592.42  4983.2  591.59  4983.7  591.09
  4995.5  591.59  5009.6  593.56    5040  592.81  5071.4  594.65  5110.8  594.89
  5180.5  597.49  5234.3  600.22  5267.3  601.75  5302.9   605.8  5331.3  605.79
  5343.4  606.58    5454  608.08  5608.7  608.61  5700.4  608.59  5738.2  608.54
#Mann= 11 ,-1 , 0
  3554.4     .05       0  3945.9    .045       0  4798.3     .07       0
  4983.2     .05       0  4995.5     .07       0  5180.5    .035       0
  5234.3     .07       0  5331.3    .035       0    5454    .045       0
  5608.7    .035       0  5700.4    .045       0
Bank Sta=4983.2,4995.5
XS Rating Curve= 0 ,0
Exp/Cntr=0.3,0.1

Type RM Length L Ch R = 1 ,82266   ,441,441,441
BEGIN DESCRIPTION:
A18957
END DESCRIPTION:
XS GIS Cut Line= 3
      2287744.18     13794079.93       2287781.3      13792440.6
      2287527.78     13791939.76
#Sta/Elev= 30
  3599.9  598.14  3864.9  598.41  4294.4  596.71  4655.1  594.22  4855.2  591.93
  4915.2  592.48    4939  591.07  4939.5  590.57  4950.9  590.57  4951.4  591.07
  4975.2  592.22  5016.6  591.89  5035.2  591.21  5045.2  592.71  5055.2  593.39
  5165.2  597.06  5180.2  598.58  5186.3  599.86  5205.2  601.08  5225.2  600.57
    5247  601.99    5297  603.27  5321.7   604.1  5330.5  604.64  5436.3  606.05
  5447.7  607.21  5464.2  607.52  5503.2   607.2  5646.9  608.23    5801  608.23
#Mann= 7 ,-1 , 0
  3599.9     .05       0    4939     .05       0  4951.4     .05       0
  5016.6    .035       0    5297     .05       0  5321.7    .035       0
  5646.9    .045       0
Bank Sta=4939,4951.4
XS Rating Curve= 0 ,0
Exp/Cntr=0.3,0.1

Type RM Length L Ch R = 1 ,81825   ,426,426,426
BEGIN DESCRIPTION:
A18956
END DESCRIPTION:
XS GIS Cut Line= 3
       2287867.9     13794073.78       2288140.1     13792898.38
      2288158.66     13791920.96
#Sta/Elev= 30
  3720.2  599.04  3975.6  598.32  4563.6  593.51  4638.9  592.99    4883  590.88
  4970.1   590.9  4993.9  589.64  4994.4  589.14  5005.8  589.14  5006.3  589.64
  5030.1  590.01  5040.1  591.17  5077.1  591.25  5120.1  591.47  5290.1   594.6
  5330.2  596.48  5340.2   597.7  5360.2  597.81  5370.2  597.07  5390.2  598.26
  5414.7  598.35  5490.2  599.68  5530.2   601.6  5560.2  600.76  5642.6  601.92
  5720.2  602.69  5740.2  603.79  5755.9  603.28  5780.2  602.46  5904.3  603.46
#Mann= 9 ,-1 , 0
  3720.2     .05       0  4563.6    .035       0  4638.9     .05       0
  4993.9     .05       0  5006.3     .05       0  5077.1     .07       0
  5414.7     .05       0  5642.6    .035       0  5755.9    .045       0
Bank Sta=4993.9,5006.3
XS Rating Curve= 0 ,0
Exp/Cntr=0.3,0.1

Type RM Length L Ch R = 1 ,81399   ,408,408,408
BEGIN DESCRIPTION:
A18955
END DESCRIPTION:
XS GIS Cut Line= 3
      2287960.67     13794092.38      2288449.41     13793306.68
      2288659.75     13791964.26
#Sta/Elev= 30
  3789.1  599.39  4080.4  597.85  4152.3  596.12  4435.2  593.28  4516.7  592.57
  4755.9  591.26  4907.7  590.91  5003.3   589.3  5003.8   588.8  5015.9   589.3
    5121  590.94  5202.6  590.38  5236.2  590.28  5342.3  592.65  5485.4  595.36
  5515.7  596.76  5525.9  596.44  5546.1  598.18  5639.8   598.4  5728.3  599.23
  5752.7  600.58  5778.9  599.42  5838.1  600.46  5883.1  600.72  5910.5  601.84
  5930.7  600.75  5973.7  601.66  6042.1  602.11  6062.3  603.36  6073.2  602.86
#Mann= 11 ,-1 , 0
  3789.1     .05       0  4435.2    .035       0  4516.7     .05       0
  4755.9    .035       0  5003.3    .035       0  5015.9    .035       0
  5202.6     .05       0  5342.3    .035       0  5639.8     .05       0
  5838.1    .035       0  5973.7    .045       0
Bank Sta=5003.3,5015.9
XS Rating Curve= 0 ,0
Exp/Cntr=0.3,0.1

Type RM Length L Ch R = 1 ,80991   ,431,431,431
BEGIN DESCRIPTION:
A18954
END DESCRIPTION:
XS GIS Cut Line= 4
      2288028.75     13794098.52      2288832.96     13793572.69
      2288888.64     13792780.84      2288907.15     13792108.26
#Sta/Elev= 30
  3497.4  599.69  3620.5  599.43  3743.8  597.86  3756.1  596.76  3822.6  594.84
  3828.5  595.41  3937.1  593.12  4372.6  591.23  4591.6   590.8  4593.5   590.8
  4847.8  590.35    4887  591.56  4921.4  590.59    4991   588.1  4991.5   587.6
  5003.6   588.1    5035  589.46  5155.5  590.08  5197.8  590.52    5238  592.39
  5453.4  598.08    5498  599.28    5538  601.52    5568  600.91    5618  602.37
  5648.1  601.48  5713.9  602.44  5788.1  603.63  5828.3  602.95  5924.9  603.47
#Mann= 13 ,-1 , 0
  3497.4     .05       0  4372.6    .035       0  4591.6     .05       0
  4593.5    .035       0  4921.4     .05       0    4991     .05       0
  5003.6     .05       0    5035    .035       0  5155.5     .05       0
    5238     .07       0  5453.4    .035       0  5713.9     .05       0
  5828.3    .035       0
Bank Sta=4991,5003.6
XS Rating Curve= 0 ,0
Exp/Cntr=0.3,0.1

Type RM Length L Ch R = 1 ,80560   ,383,383,383
BEGIN DESCRIPTION:
A18953
END DESCRIPTION:
XS GIS Cut Line= 4
      2288078.23     13794117.08      2289148.46     13793442.77
      2289346.43      13792756.1      2289433.03     13792242.64
#Sta/Elev= 30
    3300  600.05  3423.1  599.58  3517.2  597.91  3594.4  595.15    3615  594.55
  3773.9  592.63  3874.4  592.26    4117  591.27    4313  590.61  4336.3  592.13
  4439.6   590.3  4958.1  588.59  4970.7  588.23    4998  584.49  4998.5  583.99
  5010.6  584.49  5020.5  586.87    5038  588.51  5115.7  589.41    5183  591.66
  5221.9  590.88  5298.5  594.42  5341.5  593.69  5419.5     597    5443   595.9
  5534.2  599.78  5564.7  598.87  5655.9  602.39  5696.5  601.26  5800.3  603.89
#Mann= 9 ,-1 , 0
    3300     .05       0  3594.4    .035       0    3615     .05       0
  3773.9    .035       0  3874.4     .05       0    4117    .035       0
  4439.6     .05       0    4998     .05       0  5010.6     .05       0
Bank Sta=4998,5010.6
XS Rating Curve= 0 ,0
Exp/Cntr=0.3,0.1

Type RM Length L Ch R = 1 ,80177   ,962,962,962
BEGIN DESCRIPTION:
A18952
END DESCRIPTION:
XS GIS Cut Line= 4
      2288109.13     13794154.22      2289507.27     13793368.54
       2289717.6     13792947.87       2289717.6     13792180.76
#Sta/Elev= 30
  3201.8  600.69  3320.6  599.16  3420.9  597.57  3523.5  594.24  3681.2  592.85
  3843.6  591.94  3973.5  591.49  4152.1  591.07  4168.1  592.63  4189.7  591.36
  4272.5   590.7  4843.1   588.7  4969.9   587.1  5015.6  583.28  5016.1  582.78
  5028.3  583.28  5044.3  586.51  5066.7  587.38  5305.9  588.72  5408.8  589.27
  5468.8  590.86  5498.8  590.03  5575.5  591.88  5648.8  592.55  5728.8  595.63
  5768.8  595.17  5848.8  598.14  5888.8  597.79  5978.8  600.71    6043  600.34
#Mann= 12 ,-1 , 0
  3201.8    .035       0  3320.6     .05       0  3420.9    .035       0
  3523.5     .05       0  3681.2    .035       0  3843.6     .05       0
  3973.5    .035       0  4272.5     .05       0  5015.6     .05       0
  5028.3     .05       0  5305.9    .035       0  5575.5     .05       0
Bank Sta=5015.6,5028.3
XS Rating Curve= 0 ,0
Exp/Cntr=0.3,0.1

Type RM Length L Ch R = 1 ,79215   ,1143,1143,1143
BEGIN DESCRIPTION:
ALLIGATOR CREEK 94.0
END DESCRIPTION:
XS GIS Cut Line= 3
      2290883.44     13796374.25      2290388.65     13792988.85
      2290050.11     13791165.98
#Sta/Elev= 30
  1665.5   599.2  2317.9  593.98  3170.6  589.53  3797.2  589.56  4231.7  592.05
  4585.4  588.68  4767.4  584.62  4801.8   583.4    4828  580.86  4848.2   583.3
  4894.5   583.6  4969.5  583.78  4979.4  579.28  4980.4  578.78  5020.1  579.28
  5030.1  584.71  5038.9   584.8    5039   584.8  5076.5  587.54  5135.4  588.37
  5365.4  587.04  5619.7  590.24    5701  591.68  5731.6  593.53  5751.9  592.56
  5853.6  596.76  6002.8   599.4  6174.4  602.84  6246.4  601.73  6940.9  601.91
#Mann= 9 ,-1 , 0
  1665.5    .035       0  2317.9     .05       0  4894.5    .035       0
  4979.4    .035       0  5020.1    .035       0  5038.9     .07       0
    5039    .045       0  6002.8    .035       0  6246.4    .045       0
Bank Sta=4979.4,5020.1
XS Rating Curve= 0 ,0
Exp/Cntr=0.3,0.1
