--- GERONIMO TRIBUTARY 2.prj (project) ---

Proj Title=GERONIMO TRIBUTARY 2 Base Level Engineering
Current Plan=p01
Default Exp/Contr=0.3,0.1
English Units
Geom File=g01
Flow File=f01
Plan File=p01
Y Axis Title=Elevation
X Axis Title(PF)=Main Channel Distance
X Axis Title(XS)=Station
BEGIN DESCRIPTION:
GERONIMO TRIBUTARY 2
END DESCRIPTION:
DSS Export Rating Curves= 0
DSS Export Rating Curve Sorted= 0
DSS Export Volume Flow Curves= 0
DXF OffsetX= 0
DXF OffsetY= 0
DXF ScaleX= 1
DXF ScaleY= 10

--- GERONIMO TRIBUTARY 2.p01 (plan) ---

Plan Title=Multiple Run
Short Identifier=Multiple
Geom File=g01
Flow File=f01
Subcritical Flow
K Sum by GR= 0
Std Step Tol= 0.01
Critical Tol= 0.01
Num of Std Step Trials= 20
Max Error Tol= 0.3
Flow Tol Ratio= 0.001
Split Flow NTrial= 30
Split Flow Tol= 0.02
Split Flow Ratio= 0.02
Log Output Level= 0
Friction Slope Method= 1
Unsteady Friction Slope Method= 2
Unsteady Bridges Friction Slope Method= 1
Parabolic Critical Depth
Global Vel Dist=  1 , 1 , 1
Global Log Level= 0
CheckData=True
Encroach Param= -1, 0, 0, 0
BEGIN DESCRIPTION:
Multiple Run
END DESCRIPTION:

--- GERONIMO TRIBUTARY 2.f01 (steady flow) ---

Flow Title=Multiple
Number of Profiles=7
Profile Names=10-year,25-year,50-year,1pct_min,100-year,1pct_plu,500-year
River Rch & RM= GERONIMO TRIBUTA,Reach-1,16548
     585     936    1249     807    1611    3213    2654
River Rch & RM= GERONIMO TRIBUTA,Reach-1,15569
     701    1132    1520     987    1969    3929    3278
River Rch & RM= GERONIMO TRIBUTA,Reach-1,13363
     781    1265    1703    1108    2211    4413    3696
River Rch & RM= GERONIMO TRIBUTA,Reach-1,7827
    1131    1872    2556    1685    3363    6710    5773
River Rch & RM= GERONIMO TRIBUTA,Reach-1,5974
    1354    2258    3098    2052    4093    8168    7088
Boundary for River Rch & Prof#=GERONIMO TRIBUTA,Reach-1,1
Up Type=0
Dn Type=3
Dn Slope=0.005
Boundary for River Rch & Prof#=GERONIMO TRIBUTA,Reach-1,2
Up Type=0
Dn Type=3
Dn Slope=0.005
Boundary for River Rch & Prof#=GERONIMO TRIBUTA,Reach-1,3
Up Type=0
Dn Type=3
Dn Slope=0.005
Boundary for River Rch & Prof#=GERONIMO TRIBUTA,Reach-1,4
Up Type=0
Dn Type=3
Dn Slope=0.005
Boundary for River Rch & Prof#=GERONIMO TRIBUTA,Reach-1,5
Up Type=0
Dn Type=3
Dn Slope=0.005
Boundary for River Rch & Prof#=GERONIMO TRIBUTA,Reach-1,6
Up Type=0
Dn Type=3
Dn Slope=0.005
Boundary for River Rch & Prof#=GERONIMO TRIBUTA,Reach-1,7
Up Type=0
Dn Type=3
Dn Slope=0.005

--- GERONIMO TRIBUTARY 2.g01 (geometry) ---

Geom Title=Existing Conditions
Program Version=4.10

River Reach=GERONIMO TRIBUTA,Reach-1
Reach XY= 30
        2311725.       13768375.      2311526.05     13768064.57
      2311532.75     13767375.09      2311767.25     13767171.97
      2311172.08     13765482.98      2310982.59     13765378.35
      2311071.57     13765026.22      2310724.86     13764859.59
      2310923.39     13764668.97      2310826.04     13764335.11
      2311015.85     13764231.77      2311117.69      13763624.9
      2310580.04     13763219.92      2310576.05     13762985.43
      2310735.64     13762825.55      2310931.69     13762917.55
      2310980.67     13762726.88      2311202.18     13762799.21
      2311167.31     13762371.33      2310630.73     13761827.55
      2310464.37       13761165.      2309551.18     13760551.87
      2309419.48     13760022.56      2309175.53     13759864.55
      2309177.05     13759230.84      2309666.16     13758881.95
      2309717.47     13758124.99      2309275.74     13757735.69
      2310016.01     13757132.07        2309825.       13756775.

Type RM Length L Ch R = 1 ,16548   ,433,433,433
BEGIN DESCRIPTION:
GERONIMO TRIBUTARY 2 30.0
END DESCRIPTION:
XS GIS Cut Line= 3
      2312525.01       13768325.      2311613.07     13768272.74
      2311143.17     13768331.48
#Sta/Elev= 30
  4196.2  542.47  4282.5     540  4336.4  540.38  4376.5  538.34  4526.8  533.65
    4697  530.72  4737.4  530.73  4937.4  527.82  4975.5  525.11  4975.7  524.61
  4979.5  525.11  5027.6  527.53  5067.6  527.81  5106.2  530.35  5178.2  532.22
  5198.4  531.21  5228.6  527.74  5246.3  527.44  5268.9  529.38  5299.2  530.75
  5326.9  530.84  5331.9   531.5  5349.6  537.22  5359.6  537.14  5379.8  539.53
  5430.2   535.2  5450.3   534.6  5453.2  535.41  5470.5  539.35  5583.2  540.49
#Mann= 5 ,-1 , 0
  4196.2     .05       0  4737.4    .035       0  4975.5    .035       0
  4979.5    .035       0  5453.2     .07       0
Bank Sta=4975.5,4979.5
XS Rating Curve= 0 ,0
Exp/Cntr=0.3,0.1

Type RM Length L Ch R = 1 ,16115   ,257,257,257
BEGIN DESCRIPTION:
GERONIMO TRIBUTARY 2 29.0
END DESCRIPTION:
XS GIS Cut Line= 3
      2312174.97     13767625.01        2311525.       13767925.
      2311175.02     13768274.98
#Sta/Elev= 30
  4284.1   539.7  4471.3  533.57    4502  533.18  4515.8  533.27  4548.4  531.41
    4659  527.52  4704.9  527.48  4722.3  526.35  4727.8  526.75  4796.7  524.89
    4918  525.03  4945.4  525.05  4983.7  523.23  4983.9  522.73  4987.8  523.23
  5028.2  525.56  5077.8  526.39  5141.4  527.85  5224.3   531.3  5254.5  531.49
  5296.9  533.36  5325.2  532.75  5353.5  535.72  5367.7  534.13  5384.6  536.95
  5410.1  539.66  5452.5  535.69  5472.9  539.73  5480.8  540.84  5494.9   540.2
#Mann= 9 ,-1 , 0
  4284.1     .07       0    4502     .05       0    4918     .07       0
  4983.7     .05       0  4987.8     .07       0  5077.8    .035       0
  5224.3    .063       0  5384.6    .035       0  5472.9     .07       0
Bank Sta=4983.7,4987.8
XS Rating Curve= 0 ,0
Exp/Cntr=0.3,0.1

Type RM Length L Ch R = 1 ,15858   ,289,289,289
BEGIN DESCRIPTION:
A19032
END DESCRIPTION:
XS GIS Cut Line= 3
      2312159.34     13767597.28       2311295.9     13767697.13
      2310790.81     13767973.17
#Sta/Elev= 30
  4369.1  539.25  4479.2  536.28  4506.5  535.63  4563.3  535.14  4615.1   531.9
  4635.2  531.96  4824.7  524.65  4876.8  523.56  4927.1  524.53  4975.4   522.6
  4975.7   522.1  4979.5   522.6  5007.7  524.62  5148.6  525.27    5209  527.16
  5266.5   527.1    5369  529.77  5391.7  529.88  5429.7   531.9  5495.1  532.46
  5501.4  533.75  5537.3  535.39  5559.8  536.14  5598.5  535.78  5620.4  533.68
  5658.3  535.51  5685.8  540.77  5739.9  537.29  5767.4  539.25  5813.9  539.23
#Mann= 8 ,-1 , 0
  4369.1     .07       0  4479.2    .035       0  4506.5     .07       0
  4975.4     .05       0  4979.5     .07       0    5369    .035       0
  5537.3    .094       0  5559.8    .035       0
Bank Sta=4975.4,4979.5
XS Rating Curve= 0 ,0
Exp/Cntr=0.3,0.1

Type RM Length L Ch R = 1 ,15569   ,219,219,219
BEGIN DESCRIPTION:
A19031
END DESCRIPTION:
XS GIS Cut Line= 4
      2312176.95     13767556.17      2311671.81     13767421.08
      2311454.49     13767421.08      2310673.29     13767609.03
#Sta/Elev= 30
  4371.5  540.17    4440  538.84  4487.4   537.5  4512.4  537.77  4547.3  536.63
  4552.4  537.12  4626.9  534.63  4735.8  531.43  4782.4  528.83  4862.5  527.92
  4981.2  524.51  4991.2  523.91  5001.2  522.31    5009  519.82  5009.3  519.32
  5013.1  519.32  5013.4  519.82  5021.2  520.83  5051.2  522.76    5214  525.62
  5265.5  525.92  5452.4  530.43  5543.2  533.64  5620.5     535  5635.7  535.92
  5657.9  536.17  5728.3  538.04    5746  539.47  5871.9  540.57  5915.2  540.28
#Mann= 7 ,-1 , 0
  4371.5     .07       0    4440    .035       0  4626.9     .07       0
    5009     .05       0  5013.4     .07       0  5620.5    .035       0
  5657.9    .094       0
Bank Sta=5009,5013.4
XS Rating Curve= 0 ,0
Exp/Cntr=0.3,0.1

Type RM Length L Ch R = 1 ,15350   ,536,536,536
BEGIN DESCRIPTION:
GERONIMO TRIBUTARY 2 28.0
END DESCRIPTION:
XS GIS Cut Line= 3
       2312147.6     13767468.08      2311554.34      13767215.5
      2310774.98       13767175.
#Sta/Elev= 30
  4415.9  539.78  4564.8  537.89  4793.8   530.4  4817.4   530.8  4853.5  533.01
  4922.8  533.57  4970.1  532.66  4975.5  530.64  4993.7  528.61  4999.2  525.92
  5016.5  523.28  5022.8   521.4  5028.2  523.88  5038.2  520.79  5044.2  519.99
  5044.5  519.49  5048.6  519.99  5051.9  529.39  5057.6  530.15  5165.9  532.43
  5220.2  528.04  5240.3  525.95  5250.3  523.32  5260.3  523.24  5480.6  528.58
  5530.7  530.45  5548.9  532.35  5560.7  534.67  5620.8  539.35  5841.1     552
#Mann= 3 ,-1 , 0
  4415.9    .035       0  5044.2    .035       0  5048.6    .035       0
Bank Sta=5044.2,5048.6
XS Rating Curve= 0 ,0
Exp/Cntr=0.3,0.1

Type RM Length L Ch R = 1 ,14814   ,290,290,290
BEGIN DESCRIPTION:
GERONIMO TRIBUTARY 2 27.0
END DESCRIPTION:
XS GIS Cut Line= 3
      2312588.05     13766980.56        2311384.     13766892.45
      2310555.86     13767009.92
#Sta/Elev= 30
  3963.4  544.68  4015.5  543.21  4066.7  540.45  4104.9  540.21  4116.9   539.4
  4319.3  536.93    4516  534.15  4808.7  524.98  4939.1  523.59  4979.2  521.93
    4997  519.33  4997.3  518.83  5001.5  519.33  5049.3  520.02  5089.5  522.74
  5172.7  526.01  5224.8  529.16  5270.7  532.95  5295.8  534.04  5321.2  536.33
  5432.5  537.51  5452.5  538.73  5508.6  538.23  5513.7   540.6  5579.6  541.64
  5584.6  543.88  5650.5  545.65  5655.6  546.83  5664.6   547.2  6007.1  558.08
#Mann= 6 ,-1 , 0
  3963.4    .094       0  4015.5    .063       0  4319.3    .035       0
    4997    .035       0  5001.5    .035       0  5432.5    .063       0
Bank Sta=4997,5001.5
XS Rating Curve= 0 ,0
Exp/Cntr=0.3,0.1

Type RM Length L Ch R = 1 ,14524   ,320,320,320
BEGIN DESCRIPTION:
GERONIMO TRIBUTARY 2 26.0
END DESCRIPTION:
XS GIS Cut Line= 3
      2312323.79     13766757.37      2311636.57     13766645.76
      2310544.07     13766587.03
#Sta/Elev= 30
  4155.5  535.12  4215.1  533.35  4245.5  530.56  4323.8  532.17  4374.8  530.32
  4397.4     530    4447   527.4  4452.1  528.04  4488.6   526.1  4508.6  526.57
  4513.7  525.88  4539.3   527.2  4569.6  527.33  4667.7  525.43  4943.4  521.73
  4963.8  521.06  4983.5  518.17  5001.2  518.06  5001.5  517.56  5005.9  518.06
  5043.6  519.25  5063.6  521.37  5083.6  525.07  5103.7  527.69  5148.8  525.36
  5173.8  522.08  5484.6     527  5701.9  531.74  5890.1  538.42  5945.8  538.54
#Mann= 7 ,-1 , 0
  4155.5    .035       0  4374.8     .07       0  4667.7    .035       0
  5001.2    .035       0  5005.9    .035       0  5148.8     .07       0
  5484.6    .035       0
Bank Sta=5001.2,5005.9
XS Rating Curve= 0 ,0
Exp/Cntr=0.3,0.1

Type RM Length L Ch R = 1 ,14204   ,375,375,375
BEGIN DESCRIPTION:
GERONIMO TRIBUTARY 2 25.0
END DESCRIPTION:
XS GIS Cut Line= 3
      2312200.43     13766199.37      2311360.51     13766340.34
      2310749.78     13766275.74
#Sta/Elev= 30
  4258.6  541.23  4411.1  538.64  4495.3  538.17    4548  534.46  4588.6  534.75
  4691.8   530.8  4730.5  529.41  4749.4  527.79  4801.3  523.97  4872.5  521.22
  4943.5  520.52  4988.2  519.07    5002  515.14  5002.3  514.64  5006.3  514.64
  5006.7  515.14  5014.5  515.52  5024.6  518.86  5075.3  520.01  5085.4   519.5
  5117.2  520.04    5146  521.26  5196.3  520.81  5400.6  523.67  5447.6   525.2
  5457.7   524.8    5518  527.19  5638.7  528.99  5709.1  531.36  5724.4  532.45
#Mann= 8 ,-1 , 0
  4258.6    .035       0  4411.1     .07       0  4495.3    .063       0
  4691.8    .035       0  4749.4     .12       0    5002     .05       0
  5006.7     .12       0  5196.3    .035       0
Bank Sta=5002,5006.7
XS Rating Curve= 0 ,0
Exp/Cntr=0.3,0.1

Type RM Length L Ch R = 1 ,13829   ,466,466,466
BEGIN DESCRIPTION:
GERONIMO TRIBUTARY 2 24.0
END DESCRIPTION:
XS GIS Cut Line= 3
      2311675.03       13766075.        2311275.       13766025.
      2310875.05       13766025.
#Sta/Elev= 30
  4597.2   529.6  4657.7  526.52  4677.9  525.07  4708.1  523.52  4728.2  521.83
  4788.7  520.77  4808.9  519.92  4876.9   518.3  4899.6  518.56    4950  518.03
  4957.5  517.42  4970.1  517.67  4980.2  517.04  4987.9   512.9  4988.2   512.4
  4992.3   512.4  4992.7   512.9  4997.8  515.43  5002.8  515.43  5010.3  517.81
  5020.3  518.78  5030.3  518.94  5040.3  518.29  5070.3  519.18  5180.3  521.08
  5220.3  522.14  5330.3  526.06  5360.3  527.51  5390.3  528.24  5400.3  528.98
#Mann= 3 ,-1 , 0
  4597.2    .035       0  4987.9    .035       0  4992.7    .035       0
Bank Sta=4987.9,4992.7
XS Rating Curve= 0 ,0
Exp/Cntr=0.3,0.1

Type RM Length L Ch R = 1 ,13363   ,447,447,447
BEGIN DESCRIPTION:
GERONIMO TRIBUTARY 2 23.0
END DESCRIPTION:
XS GIS Cut Line= 3
      2311574.99       13765575.        2311175.       13765625.
      2310924.96     13765725.02
#Sta/Elev= 30
  4590.7  527.95  4593.2  527.95  4600.8  526.76  4628.5  524.45  4701.5  521.72
  4822.5  518.79  4842.6  517.91  4870.3  517.84  4963.6  515.83  4973.6  516.38
  4983.7  516.25  4996.5   515.7  5003.2  510.13  5006.2  509.98  5006.5  509.48
  5010.7  509.48  5011.1  509.98  5026.1  515.77  5032.8   516.4  5062.5  516.63
  5092.1  518.22  5116.3  518.87    5123  519.51  5133.8  519.85  5155.4  521.59
    5172  522.27  5184.2  522.67  5209.2  523.12  5230.7  524.52  5263.1   524.9
#Mann= 5 ,-1 , 0
  4590.7     .12       0  5006.2     .05       0  5011.1     .12       0
    5172    .035       0  5184.2     .12       0
#XS Ineff= 2 , 0
       0  4884.4  523.28               0
Permanent Ineff=
       F       F
Bank Sta=5006.2,5011.1
XS Rating Curve= 0 ,0
Exp/Cntr=0.3,0.1

Type RM Length L Ch R = 1 ,12916   ,486,486,486
BEGIN DESCRIPTION:
GERONIMO TRIBUTARY 2 22.0
END DESCRIPTION:
XS GIS Cut Line= 3
      2311425.02     13765124.99        2311025.       13765325.
      2310675.02     13765474.99
#Sta/Elev= 30
  4552.4  526.03  4611.1  524.17  4633.5  522.62  4650.2  522.76  4664.2  521.98
  4678.2  520.42    4695  519.81  4762.1  517.85  4857.1  516.27  4901.8  514.42
  4905.9   513.6  4910.2  512.73  4918.6  510.07  4942.4  510.06  5017.1  510.05
  5169.1  510.38  5182.1  509.84  5182.5  509.34  5186.7  509.34  5187.1  509.84
    5219  511.07  5237.2   510.8  5242.6  513.26  5249.9  513.84  5260.7  515.63
  5271.6  519.36  5304.3  525.43  5336.9  526.72  5358.7  528.73  5380.4  528.37
#Mann= 7 ,-1 , 0
  4552.4     .07       0  4905.9     .12       0  4942.4    .033       0
  5017.1     .12       0  5169.1    .035       0  5182.1    .033       0
  5187.1    .035       0
#XS Ineff= 2 , 0
       0  4991.2  520.81               0
Permanent Ineff=
       F       F
Bank Sta=5182.1,5187.1
XS Rating Curve= 0 ,0
Exp/Cntr=0.3,0.1

Type RM Length L Ch R = 1 ,12430   ,508,508,508
BEGIN DESCRIPTION:
GERONIMO TRIBUTARY 2 21.0
END DESCRIPTION:
XS GIS Cut Line= 3
        2311325.       13764775.        2310925.       13764975.
      2310624.99     13765275.01
#Sta/Elev= 30
  4552.8  525.22  4557.6  525.37  4628.3  524.03  4678.6  520.66  4695.4  518.16
  4717.7  517.24  4723.3  516.17  4740.1  514.76  4790.4  513.26  4807.2  511.51
  4812.7  511.79  4821.1  510.94  4844.2  510.77  4961.1  510.14  4961.5  509.64
  4965.8  509.64  4966.2  510.14    4986  510.34  4991.6  511.42  5056.6  512.38
  5127.3   511.6  5212.1  511.63  5240.4  512.38  5254.6  512.95  5268.7  515.19
  5282.9  519.51  5292.9  521.14    5297  521.81  5381.9  526.12  5424.3  526.86
#Mann= 6 ,-1 , 0
  4552.8    .035       0  4557.6     .12       0  4844.2    .033       0
  4961.1    .033       0  4966.2    .033       0  5292.9     .07       0
Bank Sta=4961.1,4966.2
XS Rating Curve= 0 ,0
Exp/Cntr=0.3,0.1

Type RM Length L Ch R = 1 ,11922   ,416,416,416
BEGIN DESCRIPTION:
GERONIMO TRIBUTARY 2 20.0
END DESCRIPTION:
XS GIS Cut Line= 3
      2311430.53      13764667.6      2310809.67     13764706.12
      2310368.95     13764737.76
#Sta/Elev= 30
  4468.8   530.2  4476.9  530.12  4508.5  529.29  4554.5   525.6  4564.5  526.19
  4624.5  525.18  4664.4  524.87  4724.8  520.91  4784.9   516.3    4815   512.9
    4825   510.7  4832.8  510.41  4833.2  509.91  4837.5  509.91  4837.9  510.41
  4855.1  511.48  4872.3  511.75  4935.2  511.08  4985.3  512.46  5025.4  512.52
  5045.4   513.1  5065.5  514.93  5075.5  514.51  5168.9  518.02  5255.9  521.03
  5282.9  522.79    5296  522.81  5356.2  525.44  5386.3  525.85  5532.7  531.68
#Mann= 7 ,-1 , 0
  4468.8    .035       0  4476.9    .063       0  4624.5     .12       0
  4832.8    .033       0  4837.9     .12       0  4872.3    .033       0
  5168.9     .07       0
Bank Sta=4832.8,4837.9
XS Rating Curve= 0 ,0
Exp/Cntr=0.3,0.1

Type RM Length L Ch R = 1 ,11506   ,439,439,439
BEGIN DESCRIPTION:
GERONIMO TRIBUTARY 2 19.0
END DESCRIPTION:
XS GIS Cut Line= 3
        2311225.       13764375.        2310825.       13764325.
      2310675.02     13764275.01
#Sta/Elev= 30
  4600.7  522.53  4643.5   522.2  4661.2  520.35  4670.7  518.37  4719.1   514.5
  4761.9  512.63  4822.4  511.56  4832.5  509.57  4842.6  506.24  4852.6   505.2
  4882.8  504.99  4883.2  504.49  4887.6  504.49    4888  504.99    4893  505.83
    4903  509.24  4913.1  510.57    4966   509.2  4973.6  508.73  4983.7  506.57
  4993.7  506.67  5001.3  508.22  5006.4  508.22  5014.4  511.04    5046   513.6
  5056.5  515.44  5088.1  519.31  5119.8   521.2  5151.4  523.86  5161.9  524.16
#Mann= 4 ,-1 , 0
  4600.7    .063       0  4670.7     .12       0  4882.8     .05       0
    4888     .12       0
Bank Sta=4882.8,4888
XS Rating Curve= 0 ,0
Exp/Cntr=0.3,0.1

Type RM Length L Ch R = 1 ,11067   ,471,471,471
BEGIN DESCRIPTION:
GERONIMO TRIBUTARY 2 18.0
END DESCRIPTION:
XS GIS Cut Line= 3
      2311275.04     13764024.99        2311025.       13764075.
      2310675.05     13764124.99
#Sta/Elev= 30
    4740  523.91    4791  521.37  4811.4  519.25    4842  514.85  4872.5  512.64
  4964.4  509.13  4984.8   507.6  4992.4  506.51  4997.5  506.51  5005.1  504.95
  5012.5   504.1    5013   503.6  5017.4   503.6  5017.8   504.1  5025.3  504.77
  5035.4   504.5  5045.5  505.19  5065.7  508.75  5075.8  508.96  5085.9  508.32
  5136.4  509.84  5156.6  509.82  5173.5  510.36  5207.1  511.26  5239.4  514.46
  5273.4  516.66    5298  519.04  5308.1  519.33  5318.2   520.4  5348.5  522.16
#Mann= 7 ,-1 , 0
    4740     .12       0  4872.5      .1       0  5012.5     .05       0
  5017.8      .1       0  5173.5     .12       0  5239.4      .1       0
  5273.4     .07       0
Bank Sta=5012.5,5017.8
XS Rating Curve= 0 ,0
Exp/Cntr=0.3,0.1

Type RM Length L Ch R = 1 ,10596   ,282,282,282
BEGIN DESCRIPTION:
GERONIMO TRIBUTARY 2 17.0
END DESCRIPTION:
XS GIS Cut Line= 3
      2311224.97       13763625.        2311125.       13763625.
      2310724.98     13763975.01
#Sta/Elev= 30
  4884.8   519.1  4904.8  517.19  4924.8  514.55  4934.8  514.05  4952.1  511.73
  4974.8  508.45  4982.3  506.64  4988.1  506.64  4991.9  500.65  4995.9  499.83
  4996.3  499.33  5000.8  499.33  5001.2  499.83  5006.1  502.77  5020.4  507.34
    5027  506.92  5034.6  507.77  5041.2  506.79  5063.1  506.36  5091.1  506.12
  5119.1  506.82  5140.9  505.89  5190.3  505.97  5204.5  506.88  5239.6  507.38
  5275.7  509.26  5317.4  509.39  5422.2  512.29  5480.7  514.49  5516.3  516.38
#Mann= 5 ,-1 , 0
  4884.8     .12       0  4952.1      .1       0  4995.9     .05       0
  5001.2      .1       0  5422.2     .12       0
Bank Sta=4995.9,5001.2
XS Rating Curve= 0 ,0
Exp/Cntr=0.3,0.1

Type RM Length L Ch R = 1 ,10314   ,320,320,320
BEGIN DESCRIPTION:
A19030
END DESCRIPTION:
XS GIS Cut Line= 3
       2311389.9      13763327.2      2310961.11      13763415.3
       2310391.4     13763708.97
#Sta/Elev= 30
  4526.1  523.15  4561.7  523.52  4588.5  521.11  4654.4  518.43  4789.9  513.43
    4817  510.74  4840.3  510.96  4857.8  508.79  4957.9  504.51  4969.6  504.26
  4972.6     501    4973   500.5  4977.9     501  5013.9  501.57  5036.1  505.35
  5063.9  502.98  5102.6  505.38    5117  504.72    5252  510.53  5257.7  509.82
  5263.3  511.27  5285.7  510.74  5324.9  513.46  5340.8  515.62  5346.4  514.55
  5362.9  516.61  5368.5  515.85  5429.4  520.79  5562.4  527.22  5604.8  528.06
#Mann= 6 ,-1 , 0
  4526.1     .07       0  4654.4     .12       0  4957.9      .1       0
  4972.6     .05       0  4977.9      .1       0  5324.9     .12       0
Bank Sta=4972.6,4977.9
XS Rating Curve= 0 ,0
Exp/Cntr=0.3,0.1

Type RM Length L Ch R = 1 ,9994    ,452,452,452
BEGIN DESCRIPTION:
A19029
END DESCRIPTION:
XS GIS Cut Line= 3
      2311401.66     13763221.48       2310896.5     13763186.24
       2310239.3     13763397.48
#Sta/Elev= 30
  4287.6  523.05  4325.4  521.75  4384.5  518.38  4424.6   517.1  4474.2  514.91
  4514.8  513.74  4564.9  510.62  4629.5  507.99  4692.9   506.7  4803.5  504.77
  4840.9  504.94  4911.1  502.88  4963.6  503.35  4995.1  500.83    5004  498.21
  5004.4  497.71  5009.3  498.21  5016.1  500.36  5033.5  502.24  5102.9  504.91
  5129.8  507.78  5142.2  511.93  5167.1  516.67  5199.2  519.45  5234.3  520.93
    5324  523.63  5429.1  526.25  5436.3   527.6  5461.2  526.88  5484.3  528.61
#Mann= 10 ,-1 , 0
  4287.6     .07       0  4325.4     .12       0  4424.6     .07       0
  4474.2     .12       0  4629.5      .1       0  4692.9     .12       0
    5004     .05       0  5009.3     .12       0  5234.3     .12       0
    5324     .07       0
Bank Sta=5004,5009.3
XS Rating Curve= 0 ,0
Exp/Cntr=0.3,0.1

Type RM Length L Ch R = 1 ,9542    ,550,550,550
BEGIN DESCRIPTION:
A19028
END DESCRIPTION:
XS GIS Cut Line= 3
      2311460.34     13763080.51       2310896.5     13762998.28
      2310262.16     13762810.33
#Sta/Elev= 30
  4152.5  517.72  4218.5  516.67    4259  514.37  4269.1  515.14  4309.5  511.84
  4366.4   509.8  4428.1  508.19  4440.9   506.8  4499.5  505.23  4673.3  502.16
  4744.7  503.31  4838.6  502.21  4888.9  500.25    4922  501.26  4960.6  499.96
  4982.6  501.28  4993.8  500.83  5002.8   496.8  5003.2   496.3  5008.2   496.8
  5015.9  497.03  5026.3  500.54  5037.5  505.98  5044.1   507.1  5109.8  513.76
  5157.2  514.63  5242.2  519.35  5280.7  518.13  5313.9  520.52  5383.9  520.89
#Mann= 8 ,-1 , 0
  4152.5     .12       0  4366.4     .07       0  4428.1     .12       0
  4982.6     .07       0  5002.8     .05       0  5008.2     .07       0
  5044.1     .12       0  5157.2     .07       0
Bank Sta=5002.8,5008.2
XS Rating Curve= 0 ,0
Exp/Cntr=0.3,0.1

Type RM Length L Ch R = 1 ,8992    ,702,702,702
BEGIN DESCRIPTION:
A19027
END DESCRIPTION:
XS GIS Cut Line= 3
      2311489.68     13763062.87      2310849.51     13762733.97
       2310344.4     13762692.86
#Sta/Elev= 30
  4369.5  517.47  4409.5  515.11    4439  514.75  4549.9  508.86  4653.5  505.97
  4664.5  505.28  4734.5  502.83  4788.3  497.84  4832.7  500.06  4877.1  498.61
  4891.9  499.34  4899.3  498.01  4952.6  498.35  4971.4  497.19  4985.3  493.83
  4985.7  493.33  4990.7  493.83  4993.6  498.12  5033.1  499.23  5103.8  500.71
    5174  506.94    5197  506.36  5217.9  507.16  5314.5  510.54  5344.6  510.31
  5374.7     512  5394.7  511.49  5497.9  514.21  5575.3  516.29    5596   515.4
#Mann= 11 ,-1 , 0
  4369.5     .07       0  4409.5     .12       0  4653.5     .07       0
  4664.5     .12       0  4952.6      .1       0  4985.3     .05       0
  4990.7      .1       0  5033.1     .12       0    5197     .07       0
  5217.9     .12       0  5497.9     .07       0
Bank Sta=4985.3,4990.7
XS Rating Curve= 0 ,0
Exp/Cntr=0.3,0.1

Type RM Length L Ch R = 1 ,8290    ,463,463,463
BEGIN DESCRIPTION:
GERONIMO TRIBUTARY 2 13.0
END DESCRIPTION:
XS GIS Cut Line= 3
      2311524.99     13762125.01        2311125.       13762525.
        2310825.       13762575.
#Sta/Elev= 30
  4438.4  516.12  4452.5  514.66  4494.9  512.05  4551.5  507.14  4593.9  502.24
  4681.2   497.5  4707.1  493.98  4735.4  489.22  4749.5  496.46  4763.6  497.23
  4834.4  497.99  4862.6  497.14  4876.8  495.05  4890.9  494.12  4905.1  494.65
  4933.4  493.03  4975.8  492.22  4986.5   488.1  4987.2  487.83  4987.6  487.33
  4992.2  487.33  4992.7  487.83  5000.5  498.55  5014.2   499.1  5158.7  499.99
  5166.3   500.5  5237.2  501.49  5247.4   502.4  5280.3  502.36  5308.2  503.26
#Mann= 5 ,-1 , 0
  4438.4     .12       0  4681.2      .1       0  4986.5     .12       0
  4987.2     .05       0  4992.7     .12       0
Bank Sta=4987.2,4992.7
XS Rating Curve= 0 ,0
Exp/Cntr=0.3,0.1

Type RM Length L Ch R = 1 ,7827    ,470,470,470
BEGIN DESCRIPTION:
GERONIMO TRIBUTARY 2 12.0
END DESCRIPTION:
XS GIS Cut Line= 3
      2311125.01     13762024.99        2310975.       13762175.
        2310775.       13762375.
#Sta/Elev= 30
  4787.4  503.65    4791  503.65  4815.7     501    4844  499.77  4858.1  498.98
  4913.7  495.39  4928.8  494.24    4943   494.7  4957.1  494.26  4971.3  493.01
  4985.4   490.4    4996  487.16  5003.1  487.16  5009.9  486.53  5010.4  486.03
  5016.9  486.03  5017.4  486.53  5027.8  492.65    5042  494.03  5056.1  494.11
  5094.9  495.17  5101.6  495.33    5141   496.7  5155.1  498.24  5169.3  498.33
  5230.9  499.76  5245.1  500.34  5268.3  501.57  5278.9  500.83  5282.4  500.83
#Mann= 8 ,-1 , 0
  4787.4     .07       0  4913.7      .1       0  5009.9     .05       0
  5017.4      .1       0  5094.9     .12       0  5101.6     .05       0
  5230.9     .07       0  5245.1     .05       0
Bank Sta=5009.9,5017.4
XS Rating Curve= 0 ,0
Exp/Cntr=0.3,0.1

Type RM Length L Ch R = 1 ,7357    ,193,193,193
BEGIN DESCRIPTION:
GERONIMO TRIBUTARY 2 11.0
END DESCRIPTION:
XS GIS Cut Line= 3
      2310875.02     13761724.98        2310675.       13761875.
      2310524.97     13762025.03
#Sta/Elev= 30
    4755  499.67  4797.7   497.6  4826.9  495.75    4855  494.57  4862.3  493.95
  4891.5  492.92  4941.5  492.34  4951.5  491.79  4952.7   491.7  4968.6   489.1
  4983.2  488.69  4991.5  489.52  4997.7  488.97  5001.9  488.16  5008.6  488.16
  5019.2  486.39  5033.3  486.35  5043.7  484.13  5044.2  483.63  5050.8  483.63
  5051.3  484.13  5061.6  495.74  5075.7  496.96  5087.5  497.19    5104  497.51
  5132.3  497.36  5160.6   497.9  5188.9  499.31    5203  498.88  5217.2  499.03
#Mann= 6 ,-1 , 0
    4755     .07       0  4951.5     .05       0  4952.7     .07       0
  5043.7     .05       0  5051.3     .07       0  5087.5     .05       0
Bank Sta=5043.7,5051.3
XS Rating Curve= 0 ,0
Exp/Cntr=0.3,0.1

Type RM Length L Ch R = 1 ,7164    ,268,268,268
BEGIN DESCRIPTION:
A19026
END DESCRIPTION:
XS GIS Cut Line= 2
      2310908.25     13761426.51       2310291.5      13761966.9
#Sta/Elev= 30
  4559.8  506.97  4567.9  506.61  4582.2  507.33  4596.4  505.75  4653.3  502.33
    4696  500.51  4716.9   500.8  4731.2  499.11  4823.2  495.68  4880.2  491.98
  4949.4  491.14  4964.6  490.67  4972.2  489.21  4978.9  486.03  4986.5  483.25
  4989.3  482.92  4989.8  482.42  4996.4  482.42  4996.9  482.92  5007.3  486.66
  5014.9  491.57  5035.9  494.57  5071.7   495.1  5092.7  494.64  5135.4   495.9
  5262.6  497.69  5291.1  498.93  5297.7  499.89  5326.2  499.29  5379.8  499.93
#Mann= 6 ,-1 , 0
  4559.8     .07       0  4949.4     .05       0  4989.3     .05       0
  4996.9     .05       0  5035.9     .07       0  5071.7     .05       0
Bank Sta=4989.3,4996.9
XS Rating Curve= 0 ,0
Exp/Cntr=0.3,0.1

Type RM Length L Ch R = 1 ,6896    ,451,451,451
BEGIN DESCRIPTION:
GERONIMO TRIBUTARY 2 10.0
END DESCRIPTION:
XS GIS Cut Line= 3
      2310675.02     13761374.98        2310575.       13761475.
        2310275.       13761675.
#Sta/Elev= 30
  4849.7  497.62  4906.3  494.94  4948.7  491.65  4962.9  485.08  4971.8  485.59
    4977  485.89  4987.6  483.18  4994.1  483.18  4998.7   480.6  5004.7  483.09
  5013.7  485.49  5019.7  485.64  5027.2  483.13  5034.7  485.54  5040.7  480.46
  5049.7  480.56  5051.9  480.06  5052.4  479.56  5059.1  479.56  5059.6  480.06
  5063.3  484.41  5068.6  489.19  5070.8  491.17  5076.8   490.9  5112.8  492.16
  5232.4  493.87  5287.1  494.71  5315.6  496.58  5329.2  495.73  5351.7  496.19
#Mann= 6 ,-1 , 0
  4849.7     .07       0  4971.8     .05       0  5051.9     .05       0
  5059.6     .05       0  5068.6     .07       0  5232.4     .05       0
Bank Sta=5051.9,5059.6
XS Rating Curve= 0 ,0
Exp/Cntr=0.3,0.1

Type RM Length L Ch R = 1 ,6445    ,239,239,239
BEGIN DESCRIPTION:
GERONIMO TRIBUTARY 2 9.0
END DESCRIPTION:
XS GIS Cut Line= 3
      2310475.01     13761024.99        2310375.       13761125.
      2310125.03     13761424.96
#Sta/Elev= 30
  4863.4  498.42  4866.9  498.42  4896.3   495.6  4904.9  494.74    4920  493.95
  4948.3  491.71  4962.4  487.61  4976.6  487.49  4990.7  485.33  5001.3  481.21
  5004.8  481.21  5008.1  479.94  5008.6  479.44  5015.4  479.44  5015.9  479.94
  5018.5  480.63  5026.3  485.11  5032.8  485.87  5040.6   488.4  5047.1  488.04
  5096.6  488.81  5154.6  490.63  5174.7  490.69  5260.6  492.87  5274.9  493.54
  5281.4  493.04  5295.8  493.61  5350.7  494.41  5367.4  495.03  5395.3  494.88
#Mann= 7 ,-1 , 0
  4863.4     .07       0  4896.3     .12       0  4904.9    .035       0
  5008.1    .035       0  5015.9    .035       0  5154.6     .07       0
  5350.7     .05       0
Bank Sta=5008.1,5015.9
XS Rating Curve= 0 ,0
Exp/Cntr=0.3,0.1

Type RM Length L Ch R = 1 ,6206    ,232,232,232
BEGIN DESCRIPTION:
A19025
END DESCRIPTION:
XS GIS Cut Line= 2
      2310444.21     13760668.85      2309804.04      13761444.1
#Sta/Elev= 30
  4627.2  514.72  4652.1  513.99  4659.9  514.51  4715.9  507.53  4738.1  507.24
  4744.6  505.58  4766.8  504.63  4837.1  499.08  4907.5   490.6  4959.7  488.06
  4972.4  485.05  4979.1  484.97  4985.6  481.54  5003.9  480.36  5004.4  479.86
  5011.7  480.36  5014.2  483.05  5022.1   485.4  5036.4  486.49  5063.7  486.58
  5082.9  488.57  5106.8   490.1  5135.4  489.84  5415.5   493.5  5448.1  495.76
  5468.9  494.98  5518.4  495.58  5575.8  496.74  5604.4  498.64  5632.6  498.05
#Mann= 7 ,-1 , 0
  4627.2     .12       0  4766.8    .035       0  4959.7     .12       0
  5003.9     .05       0  5011.7     .12       0  5082.9     .07       0
  5415.5     .05       0
Bank Sta=5003.9,5011.7
XS Rating Curve= 0 ,0
Exp/Cntr=0.3,0.1

Type RM Length L Ch R = 1 ,5974    ,467,467,467
BEGIN DESCRIPTION:
GERONIMO TRIBUTARY 2 8.0
END DESCRIPTION:
XS GIS Cut Line= 3
      2310074.99     13760575.03        2310025.       13760825.
        2309625.       13761225.
#Sta/Elev= 30
  4740.3  510.69  4770.9  508.93  4791.3  506.97  4801.5  506.93  4811.7  503.27
  4821.8  500.94  4852.4  497.06  4862.6  494.42  4872.8  490.45    4883  488.58
  4913.6  486.54  4974.8   485.2    4985  484.17  4992.7  479.67  5005.4  478.98
  5005.9  478.48  5012.8  478.48  5013.3  478.98  5023.5  484.34  5063.3  487.12
  5136.6  488.82  5193.2  491.03  5207.3  490.51  5278.1  491.32  5433.6  494.41
  5447.8  495.43    5476  495.88  5490.2  495.36  5518.5  498.39  5560.9  501.53
#Mann= 4 ,-1 , 0
  4740.3     .12       0  5005.4     .05       0  5013.3     .12       0
  5063.3     .07       0
Bank Sta=5005.4,5013.3
XS Rating Curve= 0 ,0
Exp/Cntr=0.3,0.1

Type RM Length L Ch R = 1 ,5507    ,456,456,456
BEGIN DESCRIPTION:
GERONIMO TRIBUTARY 2 7.0
END DESCRIPTION:
XS GIS Cut Line= 3
      2309875.01     13760374.99        2309625.       13760625.
      2309425.02       13760675.
#Sta/Elev= 30
  4646.4  508.06  4646.7  508.06  4674.7  506.84  4688.8  504.59  4731.3  493.11
  4736.6  492.26  4759.5  489.53  4790.2  488.11  4849.9  485.33  4943.4  484.45
  4957.5  483.54  4981.8   476.2  4982.3   475.7  4989.3   475.7  4989.8   476.2
  4996.4  480.96  5002.5  480.96  5007.8  484.17  5010.3  485.69    5018  486.77
  5082.4  489.57  5105.6  491.09  5123.7  493.29    5134   495.3  5141.7  497.64
  5146.8  498.07  5154.6  500.41  5164.9   502.2  5182.9  504.76  5206.1  506.64
#Mann= 8 ,-1 , 0
  4646.4     .12       0  4646.7      .1       0  4736.6     .12       0
  4790.2      .1       0  4849.9     .12       0  4981.8     .05       0
  4989.8     .12       0  5007.8     .07       0
Bank Sta=4981.8,4989.8
XS Rating Curve= 0 ,0
Exp/Cntr=0.3,0.1

Type RM Length L Ch R = 1 ,5051    ,493,493,493
BEGIN DESCRIPTION:
GERONIMO TRIBUTARY 2 6.0
END DESCRIPTION:
XS GIS Cut Line= 3
      2309724.96     13760175.01        2309475.       13760225.
      2309274.97     13760425.03
#Sta/Elev= 30
  4745.5   505.9  4767.1  504.97  4776.1  504.07  4796.4   500.7    4827  493.37
    4858  487.75    4878  484.11  4949.4  482.17  4969.8  482.57    4980  483.13
  4990.2  483.04  4997.9  481.74  5003.9  481.74  5010.6  473.06  5011.1  472.56
  5018.1  472.56  5018.6  473.06  5028.7  475.99  5042.8  482.64  5071.1  484.41
  5127.7  484.65  5136.2  485.04  5170.1  486.05  5184.3  487.83  5198.4  490.72
  5212.5  494.63  5226.7  499.56  5240.8  503.62    5255  504.49  5283.3  504.96
#Mann= 6 ,-1 , 0
  4745.5      .1       0  4767.1     .12       0    4858      .1       0
  5010.6     .05       0  5018.6      .1       0  5136.2     .12       0
Bank Sta=5010.6,5018.6
XS Rating Curve= 0 ,0
Exp/Cntr=0.3,0.1

Type RM Length L Ch R = 1 ,4558    ,315,315,315
BEGIN DESCRIPTION:
A19024
END DESCRIPTION:
XS GIS Cut Line= 3
      2310015.49     13759834.78      2309263.65     13759864.15
       2308759.3     13760092.86
#Sta/Elev= 30
  4171.4   505.5  4197.7  504.14  4231.9  501.23    4252  498.04    4292  495.01
  4395.5  491.88  4402.2  491.68  4522.2  489.43  4559.3   487.7  4789.7  485.91
  4817.5  484.18  4888.4  482.38  4938.4  481.69    4994  478.42  5007.7  477.28
  5013.1   475.2  5026.7  473.21  5027.2  472.71  5034.8  473.21  5036.2  477.44
  5043.1  485.26  5053.8  488.46  5103.6  489.33  5163.9  491.56  5240.8  491.35
  5278.1  491.88  5284.7  492.86    5372  493.27  5460.4  492.89  5477.6  493.77
#Mann= 11 ,-1 , 0
  4171.4     .07       0  4197.7     .12       0  4395.5     .07       0
  4402.2    .035       0  4789.7     .12       0  4888.4     .07       0
    4994    .035       0  5026.7    .035       0  5034.8    .035       0
  5103.6     .07       0    5372     .05       0
Bank Sta=5026.7,5034.8
XS Rating Curve= 0 ,0
Exp/Cntr=0.3,0.1

Type RM Length L Ch R = 1 ,4243    ,293,293,293
BEGIN DESCRIPTION:
A19023
END DESCRIPTION:
XS GIS Cut Line= 3
      2310003.71     13759599.84      2309040.45     13759623.33
       2308740.9     13759870.02
#Sta/Elev= 30
  4170.7  499.93  4175.9  498.69  4189.4  498.46  4209.4  496.33  4279.4  492.28
  4309.5  493.06  4339.5  491.44  4400.1  490.12    4586  485.84  4821.6  482.77
  4877.2  481.19  4939.6  480.71  4966.9  479.45  4989.7  479.82  5001.1  478.14
  5015.6  471.04  5016.1  470.54  5023.7  471.04  5029.7  473.02  5039.7  480.35
  5065.4  483.04  5099.7  483.63  5129.5  485.76  5210.1  488.88    5360  490.07
  5380.8  490.86  5387.4  490.15  5401.6  491.31  5465.5  490.91  5522.3  492.74
#Mann= 8 ,-1 , 0
  4170.7     .12       0  4400.1     .07       0  4821.6    .035       0
  4877.2     .07       0  4966.9    .035       0  5015.6    .035       0
  5023.7    .035       0  5065.4     .07       0
Bank Sta=5015.6,5023.7
XS Rating Curve= 0 ,0
Exp/Cntr=0.3,0.1

Type RM Length L Ch R = 1 ,3950    ,422,422,422
BEGIN DESCRIPTION:
A19022
END DESCRIPTION:
XS GIS Cut Line= 2
      2309980.21     13759382.52      2308959.14      13759312.1
#Sta/Elev= 30
  4192.8  506.31  4226.2  501.35  4231.2  502.05  4248.1  499.59  4298.3  494.97
  4338.4  488.63  4374.1  485.81  4416.4   484.8  4448.6  483.95  4516.9  483.73
  4578.9  482.63  4769.4  480.68  4869.6  478.22  4939.8  478.75  4958.5  477.42
  4960.5  477.42  4969.9  474.53  4975.8  471.02  4976.3  470.52  4983.4  470.52
  4983.9  471.02  4989.9  475.83  4999.9  478.03  5009.9  477.89    5020  480.66
    5030  482.32  5060.1     484  5097.4  484.05  5190.4  485.48  5216.3  485.23
#Mann= 6 ,-1 , 0
  4192.8     .12       0  4416.4     .07       0  4958.5    .035       0
  4975.8    .035       0  4983.9    .035       0  5097.4    .045       0
Bank Sta=4975.8,4983.9
XS Rating Curve= 0 ,0
Exp/Cntr=0.3,0.1

Type RM Length L Ch R = 1 ,3528    ,473,473,473
BEGIN DESCRIPTION:
A19021
END DESCRIPTION:
XS GIS Cut Line= 3
      2310021.38     13759171.08      2309240.15     13759024.23
      2308993.43     13759159.34
#Sta/Elev= 30
  4392.4  508.44  4470.1  507.32  4490.5  505.57  4500.6  504.52  4506.1  502.73
  4511.2  502.68  4558.6  492.02  4563.7  492.01    4582  488.42  4592.2  487.44
  4611.1  483.46  4653.3  481.34  4679.6  481.22  4726.3  479.66  4903.4  477.94
  4993.9  475.95  5009.4   471.6  5015.5  468.48    5016  467.98  5023.6  468.48
  5039.9  469.97  5046.4  469.09  5051.5  469.78  5061.4   474.5  5070.5  477.85
    5104  480.79  5204.5  481.63  5264.5  482.79    5367  482.95  5468.6  484.14
#Mann= 8 ,-1 , 0
  4392.4     .12       0  4679.6     .07       0  4903.4     .12       0
  5015.5     .05       0  5023.6     .12       0  5061.4      .1       0
  5204.5    .035       0    5367    .045       0
Bank Sta=5015.5,5023.6
XS Rating Curve= 0 ,0
Exp/Cntr=0.3,0.1

Type RM Length L Ch R = 1 ,3055    ,292,292,292
BEGIN DESCRIPTION:
A19020
END DESCRIPTION:
XS GIS Cut Line= 3
      2310150.55     13758789.29      2309246.03     13758754.04
      2309129.26     13758859.13
#Sta/Elev= 30
  4425.6   509.8  4541.2   507.8  4571.3  507.69  4581.3  508.29  4601.3  507.16
  4665.2  506.08  4671.3  504.49  4681.3  499.39  4741.4  483.33  4751.4  481.91
  4781.4  479.49  4806.5  478.25  4841.5  476.67  4911.5  474.91  4931.5  470.98
  4949.8  469.27  4977.4  465.61  4977.9  465.11  4985.2  465.11  4985.7  465.61
  4991.6  468.07  5001.6  474.66  5011.6  475.85  5031.6  475.49  5143.1  476.71
  5245.1  479.66  5381.9  481.71  5438.7  481.48  5466.7  482.15  5487.9   481.7
#Mann= 7 ,-1 , 0
  4425.6    .035       0  4806.5     .12       0  4949.8      .1       0
  4977.4     .05       0  4985.7      .1       0  5143.1     .12       0
  5245.1    .035       0
Bank Sta=4977.4,4985.7
XS Rating Curve= 0 ,0
Exp/Cntr=0.3,0.1

Type RM Length L Ch R = 1 ,2763    ,458,458,458
BEGIN DESCRIPTION:
GERONIMO TRIBUTARY 2 3.0
END DESCRIPTION:
XS GIS Cut Line= 3
      2309975.02       13758525.        2309575.       13758475.
      2309274.97     13758525.01
#Sta/Elev= 30
  4601.2  506.55  4621.4  505.68    4639  502.83  4651.6  501.79  4661.7  499.24
  4719.6  488.04  4724.7  487.81  4745.9  483.12  4772.5  477.98  4782.6  478.47
  4853.2  476.03  4903.6  476.28  4933.8  471.81  4943.9  471.28  4953.9  472.39
  4966.5  472.67  4971.4  470.34  4984.2  466.14  4997.7  464.38  4998.2  463.88
  5005.5  463.88    5006  464.38  5006.9  464.38  5014.5  469.69    5026  473.66
  5037.3  474.65  5098.1  474.78  5171.4  477.03  5275.5  478.85  5308.5  480.51
#Mann= 7 ,-1 , 0
  4601.2     .12       0  4745.9     .07       0  4971.4     .12       0
  4997.7     .05       0    5006     .12       0    5026     .07       0
  5171.4    .035       0
Bank Sta=4997.7,5006
XS Rating Curve= 0 ,0
Exp/Cntr=0.3,0.1

Type RM Length L Ch R = 1 ,2305    ,632,632,632
BEGIN DESCRIPTION:
GERONIMO TRIBUTARY 2 2.0
END DESCRIPTION:
XS GIS Cut Line= 3
      2310024.96     13758174.99        2309675.       13758075.
      2309274.98     13758275.01
#Sta/Elev= 30
  4642.4  502.01  4664.5  500.67  4698.3  496.25  4725.6  491.21  4730.4  489.54
  4746.4  486.42  4777.6  482.16  4831.9  478.65  4871.2  476.72    4944  475.15
  4950.5  474.32  4964.8  470.58  4975.2  465.53  4984.3  462.57  4989.5  463.04
  4991.8  461.35  4992.3  460.85  4999.7  460.85  5000.2  461.35  5009.2  461.57
  5014.7  464.91  5028.7  469.05  5037.1   469.7  5059.5  469.34  5073.4  471.38
  5137.8  470.62  5221.6  472.68  5305.4  473.81  5378.1  475.96  5453.6  476.88
#Mann= 6 ,-1 , 0
  4642.4     .12       0  4730.4     .07       0  4831.9     .12       0
  4991.8     .05       0  5000.2     .12       0  5137.8     .07       0
Bank Sta=4991.8,5000.2
XS Rating Curve= 0 ,0
Exp/Cntr=0.3,0.1

Type RM Length L Ch R = 1 ,1673    ,381,381,381
BEGIN DESCRIPTION:
A19019
END DESCRIPTION:
XS GIS Cut Line= 4
      2310273.86     13757779.03      2309469.22     13757779.03
      2309246.03     13757961.11      2308975.85      13758736.4
#Sta/Elev= 30
  4025.5  493.32  4064.4  492.15  4114.4  488.65  4174.4  487.84  4284.4  483.76
  4384.4  476.14  4614.4  473.46  4764.4  473.33  4890.2  469.11  4900.8  468.67
  4915.1  466.02    4923  462.36  4925.3  459.63  4925.8  459.13  4933.7  459.63
  4964.7  463.74  4972.6  463.72    4979  465.51  4986.9  465.25  5022.1  471.77
  5065.2  473.69  5230.3  475.47    5531  478.57  5618.7  479.97    5624  479.06
  5634.2  480.18  5655.1  481.09    5673  479.58  5768.1  481.19  5939.2  480.76
#Mann= 8 ,-1 , 0
  4025.5    .035       0  4890.2     .07       0  4925.3     .05       0
  4933.7     .07       0  5230.3    .035       0    5531     .07       0
  5634.2    .035       0  5768.1    .045       0
Bank Sta=4925.3,4933.7
XS Rating Curve= 0 ,0
Exp/Cntr=0.3,0.1

Type RM Length L Ch R = 1 ,1292    ,499,499,499
BEGIN DESCRIPTION:
A19018
END DESCRIPTION:
XS GIS Cut Line= 3
      2310320.87     13757638.07      2309287.14     13757555.84
      2308993.47     13758607.19
#Sta/Elev= 30
  4062.7  493.19  4088.7  492.97  4169.2  486.28  4382.2  477.85  4449.8  474.75
  4543.9  473.33  4640.4  476.65  4760.8  476.36  4790.4  474.39  4795.4  476.04
  4851.1  470.27  4971.4  467.41  4991.5  462.53  4997.3  457.47  4997.8  456.97
  5005.7  457.47  5041.7  461.88  5046.9     464  5081.8  466.26  5098.3  471.04
  5125.5  469.33  5260.9   468.9  5272.5  467.47  5277.7  469.23  5540.6  473.94
  5923.9  478.76  5995.2  478.97    6018  480.76  6145.3  480.54  6191.3  480.11
#Mann= 9 ,-1 , 0
  4062.7     .12       0  4382.2    .035       0  4997.3    .035       0
  5005.7    .035       0  5260.9     .07       0  5540.6    .035       0
  5923.9     .07       0  5995.2    .035       0  6145.3    .045       0
Bank Sta=4997.3,5005.7
XS Rating Curve= 0 ,0
Exp/Cntr=0.3,0.1

Type RM Length L Ch R = 1 ,793     ,553,553,553
BEGIN DESCRIPTION:
A19017
END DESCRIPTION:
XS GIS Cut Line= 4
      2310356.11     13757608.69      2309668.92     13757238.66
      2309293.01     13757485.35       2308981.7     13758548.51
#Sta/Elev= 30
  4324.7  493.14  4675.2  472.61  4712.1  467.27  4720.2  470.53  4725.9  463.91
  4742.1  461.04  4757.5  467.05  4818.3     470  4867.9  466.72  4895.5  459.64
  4917.4   468.8  4927.9  469.64  4977.4   466.9  4993.6   462.5  5002.7  459.35
  5011.3     456  5011.8   455.5  5019.8     456  5043.1  463.83  5101.9  469.27
  5185.3  469.67    5357   470.8  5458.3  476.46  5503.6  476.18  5528.7  471.55
  5785.4  469.17  6042.7  473.11  6438.4  478.41  6454.6   478.5  6662.6  480.21
#Mann= 15 ,-1 , 0
  4324.7     .12       0  4675.2      .1       0  4818.3     .12       0
  4993.6      .1       0  5002.7     .12       0  5011.3     .05       0
  5019.8     .12       0  5101.9     .07       0  5185.3     .12       0
    5357    .063       0  5528.7    .035       0  5785.4     .07       0
  6042.7    .035       0  6438.4     .07       0  6454.6    .035       0
Bank Sta=5011.3,5019.8
XS Rating Curve= 0 ,0
Exp/Cntr=0.3,0.1

Type RM Length L Ch R = 1 ,240     ,0,0,0
BEGIN DESCRIPTION:
A19016
END DESCRIPTION:
XS GIS Cut Line= 4
      2310638.02     13756757.04      2309868.62     13756962.61
      2309246.03     13757479.48      2308999.68     13758388.62
#Sta/Elev= 30
  4314.2  499.33  4534.7  497.47    4691  487.79  4829.5  487.96  4885.2  476.41
  4904.5  470.52  4909.6  473.37  4944.5  466.29  4984.6  466.81  5000.5  455.84
  5005.8  455.09  5006.3  454.59  5015.8  455.09  5036.8  459.84  5064.8  463.11
    5102  464.08  5278.2  469.28  5493.1  470.18  5606.3  470.31  5755.1  471.18
  5804.1  476.04  5839.5   476.6  5853.8  476.37  5886.7  470.86  6039.5  471.56
    6143   469.8  6357.3  471.71  6741.7  477.63  6819.6  478.19  6861.7  478.19
#Mann= 15 ,-1 , 0
  4314.2    .045       0    4691     .12       0  4885.2      .1       0
  5005.8     .05       0  5015.8      .1       0  5036.8     .12       0
    5102     .07       0  5493.1    .035       0  5606.3     .12       0
  5755.1    .063       0  5886.7    .035       0    6143     .07       0
  6357.3    .035       0  6741.7     .07       0  6819.6    .035       0
Bank Sta=5005.8,5015.8
XS Rating Curve= 0 ,0
Exp/Cntr=0.3,0.1

Chan Stop Cuts=-1
Use User Specified Reach Order=0
Composite Channel Slope=5
