--- Guadalupe Tributary 23.prj (project) ---

Proj Title=Guadalupe Tributary 23 Base Level Engineering
Current Plan=p01
Default Exp/Contr=0.3,0.1
English Units
Geom File=g01
Flow File=f01
Plan File=p01
Y Axis Title=Elevation
X Axis Title(PF)=Main Channel Distance
X Axis Title(XS)=Station
BEGIN DESCRIPTION:
Guadalupe Tributary 23
END DESCRIPTION:
DSS Export Rating Curves= 0
DSS Export Rating Curve Sorted= 0
DSS Export Volume Flow Curves= 0
DXF OffsetX= 0
DXF OffsetY= 0
DXF ScaleX= 1
DXF ScaleY= 10

--- Guadalupe Tributary 23.p01 (plan) ---

Plan Title=Multiple Run
Short Identifier=Multiple
Geom File=g01
Flow File=f01
Subcritical Flow
K Sum by GR= 0
Std Step Tol= 0.01
Critical Tol= 0.01
Num of Std Step Trials= 20
Max Error Tol= 0.3
Flow Tol Ratio= 0.001
Split Flow NTrial= 30
Split Flow Tol= 0.02
Split Flow Ratio= 0.02
Log Output Level= 0
Friction Slope Method= 1
Unsteady Friction Slope Method= 2
Unsteady Bridges Friction Slope Method= 1
Parabolic Critical Depth
Global Vel Dist=  1 , 1 , 1
Global Log Level= 0
CheckData=True
Encroach Param= -1, 0, 0, 0
BEGIN DESCRIPTION:
Multiple Run
END DESCRIPTION:

--- Guadalupe Tributary 23.f01 (steady flow) ---

Flow Title=Multiple
Number of Profiles=7
Profile Names=10-year,25-year,50-year,1pct_min,100-year,1pct_plu,500-year
River Rch & RM= Guadalupe Tribut,Reach-1,22786
    1218    2064    2868    1930    3852    7685    6869
River Rch & RM= Guadalupe Tribut,Reach-1,18775
    2596    4559    6487    4456    8892   17742   16545
River Rch & RM= Guadalupe Tribut,Reach-1,16942
    3445    6107    8745    6040   12052   24047   22668
River Rch & RM= Guadalupe Tribut,Reach-1,9597
    3603    6400    9176    6345   12660   25259   23864
River Rch & RM= Guadalupe Tribut,Reach-1,6858
    4605    8251   11899    8269   16500   32921   31418
River Rch & RM= Guadalupe Tribut,Reach-1,2342
    4993    8977   12978    9039   18034   35983   34492
River Rch & RM= Guadalupe Tribut,Reach-1,936
    5015    9016   13033    9077   18110   36135   34633
Boundary for River Rch & Prof#=Guadalupe Tribut,Reach-1,1
Up Type=0
Dn Type=3
Dn Slope=0.005
Boundary for River Rch & Prof#=Guadalupe Tribut,Reach-1,2
Up Type=0
Dn Type=3
Dn Slope=0.005
Boundary for River Rch & Prof#=Guadalupe Tribut,Reach-1,3
Up Type=0
Dn Type=3
Dn Slope=0.005
Boundary for River Rch & Prof#=Guadalupe Tribut,Reach-1,4
Up Type=0
Dn Type=3
Dn Slope=0.005
Boundary for River Rch & Prof#=Guadalupe Tribut,Reach-1,5
Up Type=0
Dn Type=3
Dn Slope=0.005
Boundary for River Rch & Prof#=Guadalupe Tribut,Reach-1,6
Up Type=0
Dn Type=3
Dn Slope=0.005
Boundary for River Rch & Prof#=Guadalupe Tribut,Reach-1,7
Up Type=0
Dn Type=3
Dn Slope=0.005

--- Guadalupe Tributary 23.g01 (geometry) ---

Geom Title=Existing Conditions
Program Version=4.10

River Reach=Guadalupe Tribut,Reach-1
Reach XY= 30
        2233175.     13880273.13      2233227.24     13879380.93
       2233623.8      13878714.5      2233524.79     13878145.05
      2233723.64     13877865.35      2233777.07     13876930.86
      2234223.94     13876114.56      2234077.24     13874780.93
      2234635.63       13873865.      2235022.58     13873580.54
      2235319.07     13873527.23      2235840.27     13873824.63
      2236069.64      13873727.7      2236226.99     13871730.68
      2236724.62     13871159.73      2236425.76     13870485.69
      2236530.52     13870122.57      2237021.89     13869523.35
      2236826.05     13868985.43       2237273.8      13868364.5
      2237324.49     13867640.21      2237077.07     13867069.14
      2237038.36      13866438.4      2236680.94     13866377.26
      2236063.05     13866723.07      2235340.21     13866874.49
        2234725.       13866175.      2234878.53     13864776.47
      2235461.37     13864288.21        2235575.       13863975.

Type RM Length L Ch R = 1 ,22786   ,329,329,329
BEGIN DESCRIPTION:
A19251
END DESCRIPTION:
XS GIS Cut Line= 3
      2233636.59     13880356.53      2233241.83     13880195.56
      2232555.85     13880115.08
#Sta/Elev= 30
    4506    1022  4594.1 1019.55  4601.1 1018.57  4606.5 1016.26  4630.6 1013.45
  4654.6 1014.13  4702.1 1010.14  4713.5 1007.38  4732.1 1005.77  4745.3 1002.73
  4809.7 1000.74  4863.1  998.03  4874.9  996.09  4916.6  994.43  4932.3  991.66
  4969.4  976.35  4997.6  974.08  4997.9  973.58  5001.6  974.08  5029.8  980.53
  5065.5  985.17  5153.7  989.42  5236.9  998.04  5402.3 1012.11  5432.6 1015.84
    5503  1021.5  5533.2 1022.41  5553.4 1026.82  5579.7 1030.12    5623 1033.42
#Mann= 3 ,-1 , 0
    4506     .12       0  4997.6     .05       0  5001.6     .12       0
Bank Sta=4997.6,5001.6
XS Rating Curve= 0 ,0
Exp/Cntr=0.3,0.1

Type RM Length L Ch R = 1 ,22457   ,450,450,450
BEGIN DESCRIPTION:
Guadalupe Tributary 23 46.0
END DESCRIPTION:
XS GIS Cut Line= 3
      2233851.13     13879954.13        2233225.       13879875.
      2232638.15      13879862.2
#Sta/Elev= 30
  4368.9 1041.28  4455.7  1028.5  4481.3 1020.91    4496 1020.48  4536.4  1015.4
  4556.4  1009.8  4576.7 1008.71  4636.6 1001.46  4778.3  995.45    4869  993.14
  4889.1  989.35  4929.5   985.9  4969.8   978.3  4995.5  969.78  4995.7  969.28
  4999.5  969.78    5010  970.53    5020  972.89    5130  981.51  5170.1  988.54
  5200.1  991.66  5220.1  995.86  5291.5 1001.13  5330.1 1004.52    5390 1006.88
  5450.1 1012.62  5480.1 1017.35  5510.1 1019.69  5540.1 1026.07    5587 1031.99
#Mann= 5 ,-1 , 0
  4368.9     .12       0  4995.5     .05       0  4999.5     .12       0
  5291.5     .07       0    5390     .12       0
Bank Sta=4995.5,4999.5
XS Rating Curve= 0 ,0
Exp/Cntr=0.3,0.1

Type RM Length L Ch R = 1 ,22007   ,471,471,471
BEGIN DESCRIPTION:
Guadalupe Tributary 23 45.0
END DESCRIPTION:
XS GIS Cut Line= 3
      2233717.03     13879574.75        2233225.       13879425.
      2232693.83     13879413.79
#Sta/Elev= 30
  4485.3 1003.95  4529.2 1001.36  4550.1  998.82  4568.1  998.07  4581.5  995.83
  4677.1  991.04  4759.2  985.37  4790.6  981.73  4808.5  981.25  4832.4   978.6
  4853.3  974.22  4945.1   969.3  4968.3  968.94  4987.2  964.93  4987.4  964.43
  4991.2  964.93    4997   968.7  5002.1   968.7  5009.6  971.73  5049.6   981.4
  5069.6  983.95  5099.6  989.55  5149.6  992.47  5179.7  996.55  5279.7 1003.89
  5359.7 1012.34  5389.7 1014.48  5409.7 1017.14  5419.7 1019.59  5530.9 1031.77
#Mann= 3 ,-1 , 0
  4485.3     .12       0  4987.2     .05       0  4991.2     .12       0
Bank Sta=4987.2,4991.2
XS Rating Curve= 0 ,0
Exp/Cntr=0.3,0.1

Type RM Length L Ch R = 1 ,21536   ,420,420,420
BEGIN DESCRIPTION:
Guadalupe Tributary 23 44.0
END DESCRIPTION:
XS GIS Cut Line= 3
      2233574.97     13879074.99        2233425.       13879025.
      2233125.02       13879075.
#Sta/Elev= 30
  4841.9  980.57    4884   977.5  4905.1  969.76  4915.7  966.63  4926.2  964.59
  4957.8  964.32  4968.4   964.9  4978.9  964.88  4989.4  962.51  4995.4  959.99
  4995.6  959.49  4999.1  959.49  4999.4  959.99  5002.5  959.99  5020.3  964.63
  5027.9  966.16  5032.9  965.99  5040.5  967.28  5081.1  969.62  5101.4  971.62
  5192.6  976.38  5210.3  979.12  5215.4  979.25  5233.2     982  5263.6   984.2
  5271.2  985.74  5276.2  986.01  5283.8  988.14    5294  989.88  5304.1  990.35
#Mann= 3 ,-1 , 0
  4841.9     .12       0  4995.4     .05       0  4999.4     .12       0
Bank Sta=4995.4,4999.4
XS Rating Curve= 0 ,0
Exp/Cntr=0.3,0.1

Type RM Length L Ch R = 1 ,21116   ,479,479,479
BEGIN DESCRIPTION:
Guadalupe Tributary 23 43.0
END DESCRIPTION:
XS GIS Cut Line= 3
      2233724.96     13878724.98        2233625.       13878675.
      2233224.97     13878775.01
#Sta/Elev= 30
  4888.7  983.19  4891.4  983.19  4902.6  981.46  4919.4  980.45    4925  979.23
  4955.7  970.54  4969.7  965.51  4978.1  960.94  4984.4  956.29  4984.7  955.79
  4988.2  955.79  4988.5  956.29  4992.1  956.32  4997.7  958.66    5003  958.66
  5010.8   960.1  5018.5  960.56  5059.7  961.28  5093.2   960.9  5142.2  962.82
  5155.1  962.47  5229.8  964.89  5299.4  968.32  5312.3  969.21  5348.3  972.98
  5353.5   972.6  5389.6  979.42  5394.7  979.48  5402.5  981.02  5412.8  981.81
#Mann= 3 ,-1 , 0
  4888.7     .12       0  4984.4     .05       0  4988.5     .12       0
Bank Sta=4984.4,4988.5
XS Rating Curve= 0 ,0
Exp/Cntr=0.3,0.1

Type RM Length L Ch R = 1 ,20637   ,424,424,424
BEGIN DESCRIPTION:
Guadalupe Tributary 23 42.0
END DESCRIPTION:
XS GIS Cut Line= 3
      2233875.01       13878375.        2233525.       13878225.
        2233125.       13878225.
#Sta/Elev= 30
  4625.5  990.31    4640  989.94    4669  985.31  4692.6  983.74  4701.7  981.51
  4710.7  977.89  4716.2  976.98  4723.4  973.49  4745.2  966.96  4763.3  963.65
  4821.3  959.96  4868.5  958.98  4908.4  956.45  4944.6  956.16  4962.8  953.27
  4995.2  950.44  4995.4  949.94  4999.3  950.44  5003.6  952.31  5046.3  954.11
  5056.3  955.88  5076.3  961.09  5086.3  962.07  5116.3  962.99  5246.3  970.42
  5286.3  973.47  5296.3  975.21  5326.3  976.86  5376.3  984.87  5406.3   987.6
#Mann= 3 ,-1 , 0
  4625.5     .12       0  4995.2     .05       0  4999.3     .12       0
Bank Sta=4995.2,4999.3
XS Rating Curve= 0 ,0
Exp/Cntr=0.3,0.1

Type RM Length L Ch R = 1 ,20213   ,467,467,467
BEGIN DESCRIPTION:
Guadalupe Tributary 23 41.0
END DESCRIPTION:
XS GIS Cut Line= 3
      2233925.01       13877925.        2233725.       13877875.
        2233425.       13877975.
#Sta/Elev= 30
  4788.1  976.98  4790.7  976.98  4806.2  974.69    4819  973.96  4860.3  966.99
  4870.6   964.5  4880.9  960.77  4888.6  956.82  4893.8  957.48  4901.5   953.6
  4911.8  951.32  4922.1  949.79  4971.1   947.9    4984  946.95  4991.7  945.55
  4996.9  945.55  5002.7   943.7    5003   943.2  5006.6   943.2  5006.9   943.7
  5015.4  943.96  5025.9  946.06  5057.5  948.71  5089.1  950.44  5110.2   951.2
  5131.3  952.94  5162.9  954.71  5236.7  957.59  5247.3   958.4  5310.5  961.25
#Mann= 3 ,-1 , 0
  4788.1     .12       0  5002.7     .05       0  5006.9     .12       0
Bank Sta=5002.7,5006.9
XS Rating Curve= 0 ,0
Exp/Cntr=0.3,0.1

Type RM Length L Ch R = 1 ,19746   ,404,404,404
BEGIN DESCRIPTION:
Guadalupe Tributary 23 40.0
END DESCRIPTION:
XS GIS Cut Line= 3
      2233825.03     13877525.02        2233675.       13877425.
      2233275.03       13877375.
#Sta/Elev= 30
  4823.9   952.2  4831.4  952.41  4873.5  949.41  4888.5   946.8    4896  946.62
  4924.6  943.01  4945.6  941.89  4954.6  940.39  4981.7  938.11  4996.7  937.94
  5001.2  936.77  5012.2  935.55  5012.4  935.05  5016.4  935.55  5034.4  938.05
    5042  941.16  5074.8  942.42  5122.6  946.41  5195.7  950.19  5203.3  951.84
  5208.3  951.93  5215.8  953.94    5236  955.35  5266.2  959.87  5306.5  968.92
  5326.7  972.21  5346.9  977.53  5369.5  982.11  5377.1  984.93  5407.3  987.93
#Mann= 3 ,-1 , 0
  4823.9     .12       0  5012.2     .05       0  5016.4     .12       0
Bank Sta=5012.2,5016.4
XS Rating Curve= 0 ,0
Exp/Cntr=0.3,0.1

Type RM Length L Ch R = 1 ,19342   ,341,341,341
BEGIN DESCRIPTION:
Guadalupe Tributary 23 39.0
END DESCRIPTION:
XS GIS Cut Line= 3
      2234035.11     13877386.57      2233778.34     13877056.99
      2233475.01       13876925.
#Sta/Elev= 30
  4578.4  954.09  4630.1  951.26  4707.2  949.61  4764.9  946.02  4771.3  946.52
  4814.7  945.15  4878.9  941.61  4907.9  938.41  4941.7  936.02    4964  933.11
  5000.7  931.58  5019.5  928.65  5019.8  928.15  5023.8  928.65  5038.4  931.98
  5067.3  932.41  5085.3  935.24  5130.7  938.45  5166.5  942.78  5213.4  954.55
  5228.9  955.97  5242.3  958.35  5260.2  964.22  5265.7  964.83  5289.1  971.17
  5294.6  971.63  5312.6   976.1    5318  976.25  5324.3  978.34    5327  978.34
#Mann= 3 ,-1 , 0
  4578.4     .12       0  5019.5     .05       0  5023.8     .12       0
Bank Sta=5019.5,5023.8
XS Rating Curve= 0 ,0
Exp/Cntr=0.3,0.1

Type RM Length L Ch R = 1 ,19001   ,226,226,226
BEGIN DESCRIPTION:
A19250
END DESCRIPTION:
XS GIS Cut Line= 4
      2234115.58     13877256.26      2233946.96     13876800.23
      2233885.64     13876731.25      2233433.49     13876631.62
#Sta/Elev= 30
  4475.6  948.84  4562.2  944.44  4694.5  940.19  4719.6  936.04    4750  933.17
  4952.2  928.02  4967.2  925.31  4981.4  918.99  4995.6     910  5002.3  908.11
  5014.4  907.32  5014.7  906.82  5018.7  907.32  5037.4  913.48    5045  917.71
  5050.8  926.11    5057  926.11  5059.9  933.08    5065   938.2  5075.2  940.59
  5152.4   946.7  5201.3  948.65  5228.8  951.55  5342.7  956.42  5381.3  961.46
  5386.4  960.88  5402.9  964.37  5435.2  967.22  5495.1  975.78  5517.1  976.94
#Mann= 3 ,-1 , 0
  4475.6     .12       0  5014.4     .05       0  5018.7     .12       0
Bank Sta=5014.4,5018.7
XS Rating Curve= 0 ,0
Exp/Cntr=0.3,0.1

Type RM Length L Ch R = 1 ,18775   ,392,392,392
BEGIN DESCRIPTION:
A19249
END DESCRIPTION:
XS GIS Cut Line= 3
      2234586.94     13876669.93      2233977.62     13876577.96
      2233460.24     13876577.96
#Sta/Elev= 30
  4431.2  960.45  4443.3  959.54  4493.3     951  4498.3  951.43  4562.2  944.69
  4567.2   945.6  4636.1  940.68    4686  934.46  4716.3  933.06  4768.9  928.27
  4878.1  923.82  4896.5  920.23  4901.6   920.8  4918.6  915.72  4965.4  906.22
  4970.5  906.63  4984.6  901.69  4985.1  901.19  4994.2  901.69  5019.7  903.82
  5034.3  911.64  5046.2  926.59  5051.2  926.59    5060   929.8    5090  934.53
    5170  942.02    5290  947.48    5450  957.63    5520  967.52  5564.8   971.4
#Mann= 3 ,-1 , 0
  4431.2     .12       0  4984.6     .05       0  4994.2     .12       0
Bank Sta=4984.6,4994.2
XS Rating Curve= 0 ,0
Exp/Cntr=0.3,0.1

Type RM Length L Ch R = 1 ,18383   ,487,487,487
BEGIN DESCRIPTION:
Guadalupe Tributary 23 38.0
END DESCRIPTION:
XS GIS Cut Line= 3
      2234736.38      13876309.7        2234125.       13876225.
      2233559.97     13876252.22
#Sta/Elev= 30
  4386.9   986.9  4408.5  983.66  4448.9  980.35  4469.1  975.79  4489.2  973.75
  4539.7  965.24  4610.4  959.26  4650.8  953.33  4741.6  948.12  4824.7  941.68
  4852.7  935.17    4883  918.78  4891.4  915.51  4989.2  898.58  4989.7  898.08
  4998.8  898.58  5006.6  898.74  5024.1  903.09  5034.3  910.06  5044.2  917.04
  5054.2  920.78  5084.2  923.09    5157  925.96  5234.4  927.72  5284.4  930.96
  5324.5  936.23  5394.6  938.92  5434.6  943.36  5514.7  945.55  5569.8  948.42
#Mann= 5 ,-1 , 0
  4386.9     .12       0  4989.2     .05       0  4998.8     .12       0
  5034.3     .07       0    5157     .12       0
Bank Sta=4989.2,4998.8
XS Rating Curve= 0 ,0
Exp/Cntr=0.3,0.1

Type RM Length L Ch R = 1 ,17896   ,454,454,454
BEGIN DESCRIPTION:
Guadalupe Tributary 23 37.0
END DESCRIPTION:
XS GIS Cut Line= 3
      2234747.86     13875819.18        2234225.       13875775.
      2233599.12     13876029.59
#Sta/Elev= 30
  4475.7  981.91  4488.6  980.73  4518.7  975.16  4558.9  972.22    4609  965.25
  4689.3  956.77  4709.4  953.15  4779.6  948.39    4880  937.42  4910.1  936.52
  4943.1  933.24  4970.3  928.73  4980.4  923.58  4990.4  916.48  4997.9  901.39
  5003.1  901.39  5010.3  896.51  5010.8  896.01    5020  896.51  5039.2  899.84
  5068.7  901.61  5092.7  908.68  5123.9  912.57  5151.7  915.37  5183.9  916.76
  5337.5  920.59  5378.3  921.57  5443.4  929.37  5475.4  929.78  5676.1  937.42
#Mann= 5 ,-1 , 0
  4475.7     .12       0  5010.3     .05       0    5020     .12       0
  5123.9     .07       0  5337.5     .12       0
Bank Sta=5010.3,5020
XS Rating Curve= 0 ,0
Exp/Cntr=0.3,0.1

Type RM Length L Ch R = 1 ,17442   ,500,500,500
BEGIN DESCRIPTION:
Guadalupe Tributary 23 36.0
END DESCRIPTION:
XS GIS Cut Line= 4
      2234540.98     13875255.84        2234075.       13875375.
        2233975.       13875375.      2233663.39     13875914.96
#Sta/Elev= 30
  4523.2  947.34  4560.3  945.89  4578.1  943.05  4583.2  943.78  4705.7  937.74
  4741.4  933.75  4782.2   932.9    4839  926.08  4863.9  924.53  4890.6  918.65
  4899.5  914.83  4904.7  914.82  4911.3  910.99  4940.4  899.58  4952.6  896.83
  4973.2  896.41    4989  892.95  4989.5  892.45  4998.8  892.95  5001.6   895.9
  5024.2  899.25  5044.2  908.87  5054.2     911  5094.2  913.72  5154.1  913.58
  5343.9  916.44  5514.2  919.68  5594.6  924.38  5631.9  928.77  5727.6  931.68
#Mann= 5 ,-1 , 0
  4523.2     .12       0    4989     .05       0  4998.8     .12       0
  5154.1     .07       0  5343.9     .12       0
Bank Sta=4989,4998.8
XS Rating Curve= 0 ,0
Exp/Cntr=0.3,0.1

Type RM Length L Ch R = 1 ,16942   ,471,471,471
BEGIN DESCRIPTION:
Guadalupe Tributary 23 35.0
END DESCRIPTION:
XS GIS Cut Line= 5
      2234450.81       13874875.        2234175.       13874875.
        2234075.       13874875.        2233975.       13874875.
      2233688.91       13874875.
#Sta/Elev= 30
  4624.1  921.13  4649.9  919.56  4669.9  919.18  4789.9  911.37  4829.9     908
  4859.9   907.7  4879.9  906.69  4929.9  902.27  4939.9  894.83  4949.9   891.2
  4959.9  882.01  4963.9  880.88  4964.4  880.38  4975.4  880.38  4975.9  880.88
  4989.9  882.42  4997.4  886.48  5002.4  886.48  5009.9  889.87  5019.9  891.83
  5039.9  891.51  5049.9  892.05  5079.9  898.35  5097.4  902.75  5203.3  909.64
  5229.9  910.75  5289.9   914.9  5319.9  918.33  5359.9  920.62    5386  922.95
#Mann= 4 ,-1 , 0
  4624.1     .12       0  4963.9     .05       0  4975.9     .12       0
  5203.3    .035       0
Bank Sta=4963.9,4975.9
XS Rating Curve= 0 ,0
Exp/Cntr=0.3,0.1

Type RM Length L Ch R = 1 ,16471   ,410,410,410
BEGIN DESCRIPTION:
Guadalupe Tributary 23 34.0
END DESCRIPTION:
XS GIS Cut Line= 5
      2234616.02     13874702.35        2234425.       13874575.
        2234275.       13874475.        2234225.       13874375.
      2234046.77     13874018.54
#Sta/Elev= 30
  4589.7  917.26  4646.5  912.91  4682.6  909.34  4841.8  902.11  4847.8  900.39
  4862.8  897.83  4868.9  895.01  4877.9  893.98  4904.9  884.22  4913.9  883.11
  4919.9  881.19    4935  880.57    4941  878.95    4950  878.21    4956  876.37
    4986  875.85  4986.5  875.35  4998.1  875.85  5007.9   876.2  5021.9  879.94
  5030.3   895.1  5035.9  901.84  5044.3  903.24  5119.7  902.53  5276.3  903.43
    5321  902.73  5446.8   902.7  5499.9  903.81  5505.5  905.61  5509.9  904.92
#Mann= 3 ,-1 , 0
  4589.7     .12       0    4986     .05       0  4998.1     .12       0
Bank Sta=4986,4998.1
XS Rating Curve= 0 ,0
Exp/Cntr=0.3,0.1

Type RM Length L Ch R = 1 ,16061   ,447,447,447
BEGIN DESCRIPTION:
Guadalupe Tributary 23 33.0
END DESCRIPTION:
XS GIS Cut Line= 5
      2235023.81     13874615.87        2234625.       13874175.
        2234525.       13874175.        2234375.       13874175.
      2234015.92     13873876.24
#Sta/Elev= 30
  4300.9  942.12  4321.9  940.48  4336.1  935.61  4364.5   928.7  4435.5  914.34
  4477.4  910.42  4527.4  907.58  4782.2  898.85  4817.3  900.57  4945.4  898.98
  4955.4  893.81  4985.4  872.58  5009.3  869.93  5009.8  869.43  5021.4  869.93
  5035.4  874.46  5055.4  875.76  5065.4   878.2  5095.4  893.81  5105.4  897.55
  5115.4  898.99  5528.8  903.13  5549.6  905.43  5563.9   909.3  5571.8  913.75
  5578.3  915.48  5586.1  920.36  5606.9  927.92  5609.8  930.84  5612.5  930.84
#Mann= 3 ,-1 , 0
  4300.9     .12       0  5009.3     .05       0  5021.4     .12       0
Bank Sta=5009.3,5021.4
XS Rating Curve= 0 ,0
Exp/Cntr=0.3,0.1

Type RM Length L Ch R = 1 ,15614   ,446,446,446
BEGIN DESCRIPTION:
Guadalupe Tributary 23 32.0
END DESCRIPTION:
XS GIS Cut Line= 5
      2235015.57     13874406.15        2234775.       13873925.
        2234725.       13873825.        2234675.       13873725.
       2234537.5       13873450.
#Sta/Elev= 30
  4345.9  910.68  4414.3  905.16  4584.8  897.41  4763.6  894.41  4830.7  891.15
    4881  885.49  4914.6  883.41  4920.2   881.3  4928.6  881.53  4950.9  872.23
  4986.6  867.32  4987.1  866.82    4999  867.32  5040.4  875.18  5048.7  878.65
  5054.3  879.23  5062.7  885.48  5071.1  887.84  5076.7  884.77  5085.1  888.53
  5093.5  889.63  5233.2  894.92  5308.7   901.1  5322.7   903.6  5339.4  912.48
    5345  913.11  5361.8  921.95  5384.2  929.17  5412.1  934.32  5414.9  936.52
#Mann= 3 ,-1 , 0
  4345.9     .12       0  4986.6     .05       0    4999     .12       0
Bank Sta=4986.6,4999
XS Rating Curve= 0 ,0
Exp/Cntr=0.3,0.1

Type RM Length L Ch R = 1 ,15168   ,450,450,450
BEGIN DESCRIPTION:
Guadalupe Tributary 23 31.0
END DESCRIPTION:
XS GIS Cut Line= 5
      2235426.76     13874102.64        2235175.       13873725.
        2235075.       13873575.        2235025.       13873475.
      2234979.36     13873383.72
#Sta/Elev= 30
  4365.8  929.26  4373.5  925.67  4379.5  924.46  4394.5  913.62  4400.5  911.99
  4409.5  906.69  4415.5  904.88  4430.6  896.17  4445.6  891.41  4466.6  887.72
  4502.7  886.41  4574.8   886.2  4797.1  887.26  4816.7  885.09  4848.2  883.84
  4855.7  882.66  4878.3  876.24  4891.8  874.13  4941.4  871.47  4977.4  867.72
  4986.2  865.18  4986.7  864.68  4998.6  865.18  5013.9  865.21  5022.3  866.37
  5036.3  872.69    5053  884.45  5058.6  896.08    5067   897.8  5213.8  906.45
#Mann= 3 ,-1 , 0
  4365.8     .12       0  4986.2     .05       0  4998.6     .12       0
Bank Sta=4986.2,4998.6
XS Rating Curve= 0 ,0
Exp/Cntr=0.3,0.1

Type RM Length L Ch R = 1 ,14718   ,472,472,472
BEGIN DESCRIPTION:
Guadalupe Tributary 23 30.0
END DESCRIPTION:
XS GIS Cut Line= 4
      2235624.98     13874024.96        2235475.       13873625.
        2235525.       13873525.      2235585.08     13873404.84
#Sta/Elev= 30
  4572.9  927.87  4582.6  926.89    4588  925.05  4594.2  920.65  4612.9  911.24
  4626.3  900.25  4636.9  894.98  4643.2  889.86  4648.5  889.21  4668.1  882.03
  4679.7  879.97    4814  873.67  4874.6  873.02  4893.3  869.53  4899.5  867.19
  4904.8  869.12  4924.4  865.28  4929.7  867.18    4936  864.44  4946.7  862.88
    4960  862.99    4984   859.9  4984.5   859.4  4996.5   859.9  5008.4   861.6
  5036.4  862.05  5058.8  879.72  5081.1  885.99  5114.7  886.88  5246.2  883.83
#Mann= 3 ,-1 , 0
  4572.9     .12       0    4984     .05       0  4996.5     .12       0
Bank Sta=4984,4996.5
XS Rating Curve= 0 ,0
Exp/Cntr=0.3,0.1

Type RM Length L Ch R = 1 ,14246   ,246,246,246
BEGIN DESCRIPTION:
Guadalupe Tributary 23 29.0
END DESCRIPTION:
XS GIS Cut Line= 3
      2235924.37     13874136.83        2235875.       13873825.
      2235694.46     13873385.77
#Sta/Elev= 30
  4685.1  921.17  4757.8  918.89    4775  915.28  4780.1  918.41  4808.4  913.33
  4837.4  910.92  4842.4  911.88  4869.2  908.75  4919.8  908.22  4929.9  901.01
  4940.1  889.26  4950.2  882.59  4960.3  874.25  4967.1  864.92  4972.2  865.26
  4998.3  850.64  5003.5  850.64  5003.8  849.21  5004.3  848.71  5016.3  849.21
  5039.5  853.97  5044.9  853.25  5054.9  856.04  5063.4  862.65  5068.8  862.19
  5076.5  868.77  5087.3  872.99  5098.2  875.38  5314.4  882.58  5475.7  881.71
#Mann= 3 ,-1 , 0
  4685.1     .12       0  5003.8     .05       0  5016.3     .12       0
Bank Sta=5003.8,5016.3
XS Rating Curve= 0 ,0
Exp/Cntr=0.3,0.1

Type RM Length L Ch R = 1 ,14000   ,236,236,236
BEGIN DESCRIPTION:
A19248
END DESCRIPTION:
XS GIS Cut Line= 3
      2236315.26     13873880.09      2235978.03     13873642.49
      2235794.06     13873462.36
#Sta/Elev= 30
  4705.6  941.45  4759.4  940.76  4774.2  937.28  4845.6  933.35  4875.2   927.6
  4881.3  927.63  4896.1   922.3  4902.2  921.88  4925.7   913.6  4931.8   912.6
  4938.3  900.95  4946.6   891.7  4952.8  887.08  4961.4  878.24  4967.6  873.24
    4975  861.27  4982.4  852.87  4997.2  848.42  5005.2  848.39  5005.7  847.89
  5018.2  848.39  5024.2  851.34    5039  852.13  5053.8  855.55  5068.6  862.25
  5083.4  865.98  5132.7  875.02  5182.1  874.84  5316.5  880.62  5375.6  881.22
#Mann= 3 ,-1 , 0
  4705.6     .12       0  5005.2     .05       0  5018.2     .12       0
Bank Sta=5005.2,5018.2
XS Rating Curve= 0 ,0
Exp/Cntr=0.3,0.1

Type RM Length L Ch R = 1 ,13764   ,482,482,482
BEGIN DESCRIPTION:
Guadalupe Tributary 23 28.0
END DESCRIPTION:
XS GIS Cut Line= 3
      2236275.02     13873575.01        2236075.       13873475.
      2235875.03       13873475.
#Sta/Elev= 30
  4776.8  932.93  4790.8   930.3  4807.6   928.3  4821.5  925.04  4852.3  915.73
  4866.3  913.96  4874.6  911.62  4880.2  908.44  4888.6  897.26    4897  888.07
  4902.6   888.2  4919.4   872.6    4925  871.98  4933.3  861.44  4941.7  854.34
  4947.3  854.06  4955.7   849.2  4969.7  847.51  4985.5  847.13    4986  846.63
  4998.5  847.13  5000.4  850.11  5030.4  853.45  5050.4  857.94  5070.4  867.73
  5080.4  870.57  5100.4  873.01  5140.4   875.3  5160.4  877.62  5200.4  879.81
#Mann= 3 ,-1 , 0
  4776.8     .12       0  4985.5     .05       0  4998.5     .12       0
Bank Sta=4985.5,4998.5
XS Rating Curve= 0 ,0
Exp/Cntr=0.3,0.1

Type RM Length L Ch R = 1 ,13282   ,455,455,455
BEGIN DESCRIPTION:
Guadalupe Tributary 23 27.0
END DESCRIPTION:
XS GIS Cut Line= 3
      2236275.05     13873075.01        2236075.       13873025.
        2235875.       13873025.
#Sta/Elev= 30
  4793.4  890.23    4796  890.23  4811.5  887.41  4816.6  887.73    4845  878.95
  4852.7  875.54  4857.9  875.31  4886.2  862.17    4894  857.61  4899.1  856.95
  4906.8  853.46  4927.5  851.91  4948.1  847.23  4958.4   846.2  4968.7  846.07
  4976.4  844.97  4981.6   845.3  4990.5  844.74    4991  844.24    5003  844.24
  5003.5  844.74  5019.6  845.27  5029.6  848.31  5039.6  858.33  5049.6  865.33
  5059.6  870.78  5069.6  873.83  5079.6  874.98  5099.6  875.75  5199.6  876.07
#Mann= 3 ,-1 , 0
  4793.4     .12       0  4990.5     .05       0  5003.5     .12       0
Bank Sta=4990.5,5003.5
XS Rating Curve= 0 ,0
Exp/Cntr=0.3,0.1

Type RM Length L Ch R = 1 ,12827   ,479,479,479
BEGIN DESCRIPTION:
Guadalupe Tributary 23 26.0
END DESCRIPTION:
XS GIS Cut Line= 3
      2236375.04     13872675.01        2236175.       13872625.
      2235974.95     13872675.01
#Sta/Elev= 30
  4789.5  882.91  4799.8  882.86  4820.5  881.07  4841.1  876.02  4848.8  872.85
    4854  872.73  4861.7  868.88    4872  865.25  4882.3  862.48    4890   859.4
  4895.2  859.52  4902.9     857  4923.5  853.39  4931.3  850.99  4936.4  851.21
  4954.5  846.89  4977.7  844.83  5013.7  845.44    5020  844.56  5020.5  844.06
  5032.7  844.06  5033.2  844.56  5047.2  845.08    5055  849.84  5060.1  849.55
  5067.8  856.11  5078.2  861.98  5088.5  864.65  5109.1  866.17  5201.9  868.29
#Mann= 3 ,-1 , 0
  4789.5     .12       0    5020     .05       0  5033.2     .12       0
Bank Sta=5020,5033.2
XS Rating Curve= 0 ,0
Exp/Cntr=0.3,0.1

Type RM Length L Ch R = 1 ,12348   ,444,444,444
BEGIN DESCRIPTION:
Guadalupe Tributary 23 25.0
END DESCRIPTION:
XS GIS Cut Line= 3
      2236325.03     13872325.03        2236175.       13872175.
      2235774.97     13871724.97
#Sta/Elev= 30
  4787.7  862.92  4862.2  858.04  4886.7  856.85  4900.9     853  4929.2  842.08
  4957.5   837.6  4979.1  836.38  4979.6  835.88  4992.4  836.38  5035.4  838.53
  5056.3  843.61  5106.5  848.82  5113.2  850.64  5127.4  850.81  5134.1  852.93
  5141.6  852.71  5148.3  855.24  5155.8  854.64  5162.5  857.04  5209.8  858.29
  5244.5  857.91  5282.9  859.06  5304.7  863.04  5325.6  870.32  5382.4  896.16
  5431.8  913.43  5467.7  924.02  5509.6  938.36  5580.6  955.09    5602  956.64
#Mann= 6 ,-1 , 0
  4787.7     .07       0  4862.2     .12       0  4979.1     .05       0
  4992.4     .12       0  5209.8     .07       0  5244.5     .12       0
Bank Sta=4979.1,4992.4
XS Rating Curve= 0 ,0
Exp/Cntr=0.3,0.1

Type RM Length L Ch R = 1 ,11904   ,467,467,467
BEGIN DESCRIPTION:
Guadalupe Tributary 23 24.0
END DESCRIPTION:
XS GIS Cut Line= 3
      2236375.02     13872025.03        2236225.       13871775.
      2236075.01     13871625.01
#Sta/Elev= 30
  4707.9  857.04  4744.7  856.84  4810.9  856.43  4832.3  853.84  4869.3  852.96
  4875.1  851.44  4890.6  850.21  4896.5  846.95  4906.2  846.31  4917.8  842.68
  4933.4   841.3  4948.9  840.98  4954.8  839.85  4964.5  839.92  4969.5  836.58
    4970  836.08  4982.9  836.58  4985.9  837.46  4991.7  837.57  5041.9  836.99
    5056  843.29  5070.2  854.67  5084.3  864.34  5098.5  881.02  5105.5  882.87
  5112.6  890.46  5126.8  897.33  5183.3  910.95  5208.1  916.43  5211.6  916.43
#Mann= 4 ,-1 , 0
  4707.9    .035       0  4744.7     .07       0  4969.5     .05       0
  4982.9     .12       0
Bank Sta=4969.5,4982.9
XS Rating Curve= 0 ,0
Exp/Cntr=0.3,0.1

Type RM Length L Ch R = 1 ,11437   ,475,475,475
BEGIN DESCRIPTION:
Guadalupe Tributary 23 23.0
END DESCRIPTION:
XS GIS Cut Line= 3
      2236625.01     13871675.02        2236525.       13871475.
      2236125.03       13871475.
#Sta/Elev= 30
  4776.6   851.3  4807.4  852.04  4835.3  850.79    4936  840.96  4955.5   839.6
  4963.9  838.16  4969.5  834.26  4977.9  830.51  4986.3  828.03  4990.7  827.96
  4991.2  827.46  5003.6  827.46  5004.1  827.96  5050.2  828.73  5070.2  830.33
  5080.2  831.68  5100.2  835.65  5110.2  839.03  5130.2  847.72  5140.2   849.2
  5210.2  854.68  5220.2  856.53  5230.2  858.91  5240.2  862.12  5250.2  865.96
  5270.2  876.17  5340.2  902.02  5370.2   910.8  5397.7   915.8  5400.2   915.8
#Mann= 4 ,-1 , 0
  4776.6    .035       0    4936     .12       0  4990.7     .05       0
  5004.1     .12       0
Bank Sta=4990.7,5004.1
XS Rating Curve= 0 ,0
Exp/Cntr=0.3,0.1

Type RM Length L Ch R = 1 ,10962   ,471,471,471
BEGIN DESCRIPTION:
Guadalupe Tributary 23 22.0
END DESCRIPTION:
XS GIS Cut Line= 3
      2236925.05       13871075.        2236725.       13871075.
      2236124.97     13871375.02
#Sta/Elev= 30
  4795.9  864.33  4885.9   859.2  4935.9  852.03  4955.9  845.22  4993.4  823.82
  5003.1  823.42  5003.6  822.92  5016.7  823.42  5032.3  824.53  5049.1  829.24
  5093.8   833.4  5152.5  835.84  5241.9  843.19  5367.7  848.96  5384.5  853.37
  5390.1  852.61  5406.8  857.48  5412.4  856.58  5429.2  862.32  5434.8  861.41
  5451.5  867.81  5457.1  867.01  5473.9  873.32  5479.5  872.18  5496.3  880.37
  5501.9  878.94  5518.6  885.47  5546.6  886.79  5608.1  901.48  5666.8  912.45
#Mann= 3 ,-1 , 0
  4795.9     .12       0  5003.1     .05       0  5016.7     .12       0
Bank Sta=5003.1,5016.7
XS Rating Curve= 0 ,0
Exp/Cntr=0.3,0.1

Type RM Length L Ch R = 1 ,10491   ,449,449,449
BEGIN DESCRIPTION:
Guadalupe Tributary 23 21.0
END DESCRIPTION:
XS GIS Cut Line= 3
      2236724.99       13870675.        2236525.       13870675.
      2236324.99       13870675.
#Sta/Elev= 30
    4795  844.36  4797.5  844.36    4815  842.77    4865  840.01    4895  837.45
    4905  836.18    4915  834.39    4925  831.98    4935  828.98    4945  827.54
    4985  822.59  4992.5  821.76  4997.5  821.76  5008.1  820.73  5008.6  820.23
  5021.3  820.23  5021.8  820.73    5025  821.36    5035  822.53    5045  824.62
    5065  831.42    5075  832.78    5085  834.58    5095  836.93    5115  843.13
    5135  850.21    5155  855.68    5165  857.95  5192.5  860.58    5195  860.58
#Mann= 3 ,-1 , 0
    4795     .12       0  5008.1     .05       0  5021.8     .12       0
Bank Sta=5008.1,5021.8
XS Rating Curve= 0 ,0
Exp/Cntr=0.3,0.1

Type RM Length L Ch R = 1 ,10042   ,445,445,445
BEGIN DESCRIPTION:
Guadalupe Tributary 23 20.0
END DESCRIPTION:
XS GIS Cut Line= 3
      2237075.03     13870124.99        2236475.       13870275.
      2236275.05     13870324.99
#Sta/Elev= 30
  4386.9   881.8  4446.2   868.7  4451.4  868.97  4487.4  862.35  4546.6  854.97
  4569.9  851.29  4616.3  846.94  4652.4  839.76  4657.5   840.1  4665.2  837.78
  4693.6  833.75  4733.8   831.1  4747.7  831.92    4776  827.94  4822.4  828.48
  4899.7  823.72  4946.1   825.8  4964.2  817.34  4975.4  816.74  4975.9  816.24
  4989.1  816.74    5008  818.57  5015.7  823.63  5023.4  834.15  5028.6  830.12
  5036.3  839.92  5056.9  846.24  5077.5  848.06  5105.9  854.99  5211.5  860.44
#Mann= 5 ,-1 , 0
  4386.9     .12       0  4546.6    .035       0  4733.8     .12       0
  4975.4     .05       0  4989.1     .12       0
Bank Sta=4975.4,4989.1
XS Rating Curve= 0 ,0
Exp/Cntr=0.3,0.1

Type RM Length L Ch R = 1 ,9597    ,444,444,444
BEGIN DESCRIPTION:
Guadalupe Tributary 23 19.0
END DESCRIPTION:
XS GIS Cut Line= 3
      2237325.01       13869975.        2236725.       13869925.
      2236125.01     13869325.01
#Sta/Elev= 30
  4393.1  977.43  4450.8  952.03  4455.8  952.28  4483.4  938.96  4553.7  910.23
  4583.8  895.47  4623.9  883.78    4654  872.05  4740.4  852.95  4834.6  837.59
  4854.7   827.4  4881.6  823.01  4965.1  820.28  5016.4  813.85  5016.9  813.35
  5030.6  813.85  5051.8   816.6    5080  828.85  5184.8  830.74  5326.3  835.11
  5391.2  839.62  5433.6  850.11  5447.7  851.85  5546.7  858.04  5617.4  871.91
    5674  886.09  5758.9  913.16  5801.3  929.47  5840.2  948.41  5843.7  948.41
#Mann= 7 ,-1 , 0
  4393.1     .12       0  4740.4    .035       0  4881.6     .12       0
  5016.4     .05       0  5030.6     .12       0  5184.8    .035       0
  5326.3     .12       0
Bank Sta=5016.4,5030.6
XS Rating Curve= 0 ,0
Exp/Cntr=0.3,0.1

Type RM Length L Ch R = 1 ,9153    ,437,437,437
BEGIN DESCRIPTION:
Guadalupe Tributary 23 18.0
END DESCRIPTION:
XS GIS Cut Line= 3
      2237424.97     13869924.98        2236975.       13869575.
      2236374.97     13869174.98
#Sta/Elev= 30
    4430 1007.52  4470.7   996.1  4536.7  970.36  4615.5   933.7  4694.2  899.69
    4744  885.81  4758.4  879.68  4779.3  873.67  4814.5  866.95  4843.5  858.26
  4863.6  854.59  4928.6   842.6  4936.7  838.72  4949.4  819.36  4971.2  810.61
  4971.7  810.11  4985.5  810.61  5036.1  814.99  5100.7  815.83  5117.5  819.32
  5187.8  824.24  5232.1  824.94  5425.2  831.39  5446.2   834.6  5468.3  840.99
  5476.3  844.66  5512.3  854.46  5599.5  873.71  5671.6  892.13  5721.2  908.79
#Mann= 7 ,-1 , 0
    4430     .12       0  4863.6    .035       0  4971.2    .035       0
  4985.5    .035       0  5117.5     .12       0  5232.1    .035       0
  5468.3     .12       0
Bank Sta=4971.2,4985.5
XS Rating Curve= 0 ,0
Exp/Cntr=0.3,0.1

Type RM Length L Ch R = 1 ,8716    ,464,464,464
BEGIN DESCRIPTION:
Guadalupe Tributary 23 17.0
END DESCRIPTION:
XS GIS Cut Line= 3
      2237425.04     13869575.02        2236825.       13869225.
        2236275.       13868775.
#Sta/Elev= 30
  4313.1  916.01  4385.5  895.78  4475.5  877.69  4561.6  864.62  4598.8  853.08
  4679.1  835.47  4759.3   829.2  4830.5  826.61    4861  822.51  4876.7  813.53
  4882.5  814.62  4898.2  808.88  4965.5  805.92    4966  805.42  4979.8  805.92
  4994.1  811.37  4999.9  810.27    5011  812.91  5014.9  817.86  5021.4  816.05
  5029.3  819.75  5039.2  820.58  5085.3  823.53  5128.4  829.44  5192.2  851.08
  5284.8  874.18  5363.1   896.8  5412.6  917.49    5676 1054.22  5718.4 1073.07
#Mann= 6 ,-1 , 0
  4313.1    .035       0  4475.5     .12       0  4830.5    .035       0
  4965.5    .035       0  4979.8    .035       0  5039.2     .12       0
Bank Sta=4965.5,4979.8
XS Rating Curve= 0 ,0
Exp/Cntr=0.3,0.1

Type RM Length L Ch R = 1 ,8252    ,443,443,443
BEGIN DESCRIPTION:
Guadalupe Tributary 23 16.0
END DESCRIPTION:
XS GIS Cut Line= 3
      2237524.98     13869424.98        2236975.       13868825.
      2236374.98       13868675.
#Sta/Elev= 30
  4181.7   902.1  4223.9  896.41  4231.3  892.76  4302.2  880.26  4386.7  870.14
  4457.6   855.6  4493.4  852.41  4620.4  830.53  4698.1   825.9  4860.9  820.99
  4953.4  809.26  4967.2  803.61  4967.7  803.11  4981.5  803.61  5036.8  804.84
  5054.9   810.3    5060  816.48  5067.8  822.18  5157.2  833.85  5201.8  844.37
    5225  852.09    5261  868.71  5266.2  868.52  5302.3  887.35  5307.4     887
  5315.2  892.62  5348.7  908.47  5521.3 1003.02  5590.9 1036.17  5614.1 1044.36
#Mann= 4 ,-1 , 0
  4181.7     .12       0  4967.2    .035       0  4981.5     .12       0
  5157.2     .12       0
Bank Sta=4967.2,4981.5
XS Rating Curve= 0 ,0
Exp/Cntr=0.3,0.1

Type RM Length L Ch R = 1 ,7809    ,488,488,488
BEGIN DESCRIPTION:
Guadalupe Tributary 23 15.0
END DESCRIPTION:
XS GIS Cut Line= 3
      2237487.93     13869231.66        2237225.       13868475.
      2236625.02       13868425.
#Sta/Elev= 30
  4194.4  871.14  4217.9  863.63  4254.4   857.6  4280.2  856.14    4306  850.65
  4360.2  844.58  4461.6  835.72  4656.7  830.38  4741.6  821.68  4900.2   817.4
  4948.8  808.77  4954.1  805.14  5008.3  797.53  5008.8  797.03  5022.7  797.53
  5053.1     805  5075.7  807.68  5105.8  816.15  5191.2  820.94  5299.7  824.62
  5376.8  831.58  5406.9  836.98  5414.4  842.41    5447  853.45  5487.1  873.95
  5534.8  905.54  5539.8   906.6  5587.5  950.13    5595  958.85  5597.5  958.85
#Mann= 5 ,-1 , 0
  4194.4     .12       0  5008.3     .05       0  5022.7     .12       0
  5191.2    .035       0  5299.7     .12       0
Bank Sta=5008.3,5022.7
XS Rating Curve= 0 ,0
Exp/Cntr=0.3,0.1

Type RM Length L Ch R = 1 ,7321    ,463,463,463
BEGIN DESCRIPTION:
A19247
END DESCRIPTION:
XS GIS Cut Line= 4
      2237510.91     13869193.25      2237415.11     13868078.13
      2237242.66     13867966.99      2236738.39     13867928.79
#Sta/Elev= 30
    3771  861.26  3777.9  858.87  3782.9  859.47  3789.3  857.56  3896.6  841.34
  3919.8  840.18  3939.9  836.92    3980  833.13  4015.2  831.11  4598.3  820.45
  4873.3  816.75  4889.3   815.4  4949.8  815.74  4964.2  814.99  4979.3  810.69
  4985.5  802.19  4994.5  798.67  5014.4  796.64  5014.9  796.14  5028.8  796.64
  5030.8  798.99  5051.9  802.31  5123.1  805.65  5183.1  812.58  5213.4  814.17
  5253.5  825.82  5303.6  832.45  5363.8  834.08  5514.2  842.64  5601.1  844.62
#Mann= 3 ,-1 , 0
    3771     .12       0  5014.4     .05       0  5028.8     .12       0
Bank Sta=5014.4,5028.8
XS Rating Curve= 0 ,0
Exp/Cntr=0.3,0.1

Type RM Length L Ch R = 1 ,6858    ,429,429,429
BEGIN DESCRIPTION:
Guadalupe Tributary 23 14.0
END DESCRIPTION:
XS GIS Cut Line= 3
      2237875.01     13866974.99        2237275.       13867575.
        2236975.       13867775.
#Sta/Elev= 30
    4156  943.83  4159.6  943.83  4170.2  940.13  4269.2  916.73  4311.6  905.53
  4325.7  903.28    4354  896.26  4382.3  892.19    4453   874.3  4475.2  872.32
  4509.6  867.59  4566.1  857.46  4644.3  841.71  4778.3  821.09  4834.8  816.01
  4891.4  815.23  4919.7  803.45    4948  796.92  4981.3  794.88  4981.8  794.38
  4999.6  794.88  5027.1  799.21  5105.2  803.15  5141.3  807.69  5184.8  810.72
  5213.4  810.97  5249.4  813.13    5293  819.32  5336.6  828.19  5365.1  830.04
#Mann= 5 ,-1 , 0
    4156     .12       0  4475.2    .035       0  4644.3     .12       0
  4981.3     .05       0  4999.6     .12       0
Bank Sta=4981.3,4999.6
XS Rating Curve= 0 ,0
Exp/Cntr=0.3,0.1

Type RM Length L Ch R = 1 ,6429    ,451,451,451
BEGIN DESCRIPTION:
Guadalupe Tributary 23 13.0
END DESCRIPTION:
XS GIS Cut Line= 3
      2237724.98     13866575.02        2237175.       13867175.
      2236874.95     13867225.01
#Sta/Elev= 30
    4182 1031.74    4210 1022.77    4260  997.04  4274.2  987.65  4280.9  979.02
  4295.1   967.2  4337.7  939.89  4351.9  937.86  4358.6  933.07    4366   932.1
  4372.8  925.38    4387  917.96  4394.4  917.52  4415.4  904.93  4521.4  868.39
  4634.9  836.76  4642.3  838.26  4662.9  835.35  4677.4  838.27  4762.5   824.6
  4797.7  816.28  4941.1  804.11  5014.6  792.48  5015.1  791.98    5033  792.48
  5036.5  795.04    5126  798.97  5211.3  805.43  5249.4  811.71  5300.1  812.91
#Mann= 5 ,-1 , 0
    4182     .12       0  4941.1     .07       0  5014.6     .05       0
    5033     .07       0    5126     .12       0
Bank Sta=5014.6,5033
XS Rating Curve= 0 ,0
Exp/Cntr=0.3,0.1

Type RM Length L Ch R = 1 ,5978    ,419,419,419
BEGIN DESCRIPTION:
Guadalupe Tributary 23 12.0
END DESCRIPTION:
XS GIS Cut Line= 3
        2237475.       13866225.        2237125.       13866775.
      2236738.41     13866908.75
#Sta/Elev= 30
  4342.6 1112.54  4371.4 1101.86  4444.2 1060.67  4465.4 1053.56    4475 1044.66
  4495.8 1034.67  4501.8 1037.95    4517 1022.38  4522.9 1024.73  4553.4  972.44
  4574.6  951.74  4678.6   878.6  4741.4   842.2    4793  820.45  4820.1  804.27
  4892.9  787.22  4923.4  784.38  4941.3   777.1  4941.8   776.6  4959.7   777.1
  4986.9  779.26  4991.6  783.39  5004.8  779.25  5010.1  784.48  5052.8  783.96
  5072.4  783.95  5098.3  793.07  5158.1  798.08  5191.8  809.24  5403.6  809.09
#Mann= 7 ,-1 , 0
  4342.6     .12       0    4475    .033       0  4678.6     .12       0
  4941.3     .05       0  4959.7     .12       0  5052.8     .07       0
  5158.1     .12       0
Bank Sta=4941.3,4959.7
XS Rating Curve= 0 ,0
Exp/Cntr=0.3,0.1

Type RM Length L Ch R = 1 ,5559    ,481,481,481
BEGIN DESCRIPTION:
Guadalupe Tributary 23 11.0
END DESCRIPTION:
XS GIS Cut Line= 4
      2237325.01     13866274.99        2237025.       13866425.
        2236975.       13866625.      2236779.76     13866789.84
#Sta/Elev= 30
  4660.6 1072.08    4684 1059.34  4705.3 1039.48  4719.3 1017.62  4727.7  973.96
  4741.7  955.92  4853.5  875.84  4892.6  853.05  4898.2   846.2    4915  839.23
  4920.6  832.92  4937.3  824.67  4942.9  816.92  4960.3  805.27  4965.3  798.72
    4982  787.14  4987.6  777.99  4993.2   775.1  5004.9  774.92  5005.4  774.42
  5023.3  774.92  5060.4  785.63  5078.5  785.73  5088.8  782.57  5137.8  786.28
  5142.9  787.18  5150.6  794.34  5160.9  798.93  5293.9  805.54  5457.7  805.53
#Mann= 5 ,-1 , 0
  4660.6     .12       0    4684    .033       0  4960.3     .12       0
  5004.9     .05       0  5023.3     .12       0
Bank Sta=5004.9,5023.3
XS Rating Curve= 0 ,0
Exp/Cntr=0.3,0.1

Type RM Length L Ch R = 1 ,5078    ,471,471,471
BEGIN DESCRIPTION:
Guadalupe Tributary 23 10.0
END DESCRIPTION:
XS GIS Cut Line= 4
      2236774.99     13866075.01        2236575.       13866425.
        2236675.       13866625.      2236708.05     13866691.09
#Sta/Elev= 30
  4596.9 1063.38  4610.1    1063  4619.9 1060.52  4626.4 1051.99  4632.2  1055.9
  4642.2 1045.25    4648 1044.25  4654.5 1034.99  4669.6 1012.09  4677.5  970.89
  4685.4  950.51  4691.2   950.9    4707  933.58  4728.6  926.17  4735.1  917.85
  4768.6  895.16  4868.3  836.24  4889.9  829.39  4905.7  815.63  4911.5  815.54
  4927.3  800.03  4933.1  800.95  4948.9  788.48  4982.9  773.84  4983.4  773.34
  5001.3  773.84    5014  778.99  5089.4  782.49  5209.6  799.26  5297.5  802.67
#Mann= 5 ,-1 , 0
  4596.9     .12       0  4610.1    .033       0  4768.6     .12       0
  4982.9     .05       0  5001.3     .12       0
Bank Sta=4982.9,5001.3
XS Rating Curve= 0 ,0
Exp/Cntr=0.3,0.1

Type RM Length L Ch R = 1 ,4607    ,467,467,467
BEGIN DESCRIPTION:
Guadalupe Tributary 23 9.0
END DESCRIPTION:
XS GIS Cut Line= 4
        2236325.       13866025.        2236175.       13866625.
        2236325.       13866775.      2236379.38     13866829.38
#Sta/Elev= 30
  4376.5 1060.21  4510.5  986.09  4559.5  955.43  4600.7  932.45  4605.8   931.8
  4683.2  881.54  4688.3  882.97  4724.4  861.33  4729.5  863.09  4765.6  847.87
  4770.8  850.65  4806.8  838.44    4812  840.47  4848.1  822.42  4853.2  826.01
  4881.6  803.47  4889.3  792.88  4894.5  801.86  4902.2  792.81  4912.5  774.43
  4983.2  770.69  4983.7  770.19  5001.6  770.69  5037.4  778.43  5051.5  776.07
    5094  777.73  5136.4  790.08  5164.7  793.75  5283.8  798.61    5284  798.61
#Mann= 4 ,-1 , 0
  4376.5     .12       0  4983.2     .05       0  5001.6     .12       0
  5283.8    .035       0
Bank Sta=4983.2,5001.6
XS Rating Curve= 0 ,0
Exp/Cntr=0.3,0.1

Type RM Length L Ch R = 1 ,4140    ,478,478,478
BEGIN DESCRIPTION:
Guadalupe Tributary 23 8.0
END DESCRIPTION:
XS GIS Cut Line= 4
      2236024.99     13866175.01        2235775.       13866775.
        2235775.       13866975.        2235775.     13867071.21
#Sta/Elev= 30
  4345.4  923.68  4367.1  913.42  4431.5  894.97  4466.2  881.93  4497.1  874.12
  4572.9  857.88  4713.7  834.29  4779.3  819.46    4880  802.13  4897.9  796.46
  4903.8  791.64  4909.3  792.93  4921.4  787.51  4927.7  784.54  4933.1   785.2
  4951.5  776.23  4956.9  776.96  4992.7   770.6  5026.1  769.55  5026.6  769.05
  5044.6  769.55  5055.4  773.84  5065.4  775.11  5105.8  772.01  5115.4  772.79
  5125.4  777.19  5135.4  794.26  5145.4  796.61  5245.4   803.7  5291.6  809.05
#Mann= 5 ,-1 , 0
  4345.4     .12       0  4921.4    .035       0  5026.1    .035       0
  5044.6    .035       0  5105.8     .12       0
Bank Sta=5026.1,5044.6
XS Rating Curve= 0 ,0
Exp/Cntr=0.3,0.1

Type RM Length L Ch R = 1 ,3662    ,439,439,439
BEGIN DESCRIPTION:
Guadalupe Tributary 23 7.0
END DESCRIPTION:
XS GIS Cut Line= 4
      2235924.98     13866275.02        2235325.       13866875.
        2235325.       13867075.        2235325.      13867107.7
#Sta/Elev= 30
    4156  874.89  4159.5  874.89  4191.3  866.29  4198.4  863.57    4255  850.18
  4325.7  836.78    4453  818.11    4552   809.1  4610.4  800.72  4615.6   799.2
  4679.2  793.61  4693.4  791.12  4721.7  788.18  4762.7  785.18  4848.9  779.38
  4877.2   776.4  4891.4  772.51  4933.8   766.7  4976.2  765.42  4981.1  764.17
  4981.6  763.67  4999.7  764.17    5001  767.28  5014.5  768.24  5024.5  773.03
  5034.5  780.23  5054.5  799.37  5064.5  803.13  5124.5  806.55  5237.2  816.57
#Mann= 5 ,-1 , 0
    4156     .12       0  4610.4    .035       0  4762.7     .12       0
  4981.1     .05       0  4999.7     .12       0
Bank Sta=4981.1,4999.7
XS Rating Curve= 0 ,0
Exp/Cntr=0.3,0.1

Type RM Length L Ch R = 1 ,3223    ,371,371,371
BEGIN DESCRIPTION:
Guadalupe Tributary 23 6.0
END DESCRIPTION:
XS GIS Cut Line= 3
      2235275.03     13866424.98        2235025.       13866575.
      2234975.01     13866774.97
#Sta/Elev= 30
  4699.9  799.56  4723.3   797.7  4750.5  793.65  4808.8  782.93  4830.2  777.29
  4839.9  776.15  4851.5  773.61  4882.6  770.75  4898.2  769.99  4909.8  767.71
  4919.6  767.15  4925.4   767.5  4940.9   764.9  4956.5  763.24  4968.2  762.72
  4983.7  763.75  5000.2  762.43  5000.7  761.93  5018.3  761.93  5018.8  762.43
  5022.4  766.95    5043  768.93  5050.7  772.28  5055.9  777.99  5063.6  784.02
  5073.9  788.09  5084.2  793.91    5092  795.95  5104.9  797.93  5197.6  801.35
#Mann= 3 ,-1 , 0
  4699.9     .12       0  5000.2     .05       0  5018.8     .12       0
Bank Sta=5000.2,5018.8
XS Rating Curve= 0 ,0
Exp/Cntr=0.3,0.1

Type RM Length L Ch R = 1 ,2852    ,510,510,510
BEGIN DESCRIPTION:
A19246
END DESCRIPTION:
XS GIS Cut Line= 3
      2235229.06     13866049.34      2234825.61     13866282.32
      2234734.69     13866827.81
#Sta/Elev= 30
  4539.3  815.34  4576.7  810.94  4606.5  809.29  4641.4  807.72  4657.1   804.9
  4694.1   801.8  4721.8  795.55  4759.1  783.73  4786.5  777.98  4802.2   776.8
  4839.5  770.58  4876.8  766.79  4913.5  764.49  4935.7  765.16  4957.2  762.81
    4963  765.69  4984.6  765.45  4994.3  763.77  5002.9  759.46  5018.9  759.41
  5019.4  758.91  5037.5  759.41  5041.3  762.01  5097.1  778.51  5109.3  784.98
  5149.8  792.36  5284.6  794.96  5340.4  797.62  5406.3  795.98  5558.2   800.8
#Mann= 4 ,-1 , 0
  4539.3    .035       0  4606.5     .12       0  5018.9     .05       0
  5037.5     .12       0
Bank Sta=5018.9,5037.5
XS Rating Curve= 0 ,0
Exp/Cntr=0.3,0.1

Type RM Length L Ch R = 1 ,2342    ,452,452,452
BEGIN DESCRIPTION:
Guadalupe Tributary 23 5.0
END DESCRIPTION:
XS GIS Cut Line= 3
      2235074.98     13865974.99        2234675.       13865825.
      2234475.04     13865874.99
#Sta/Elev= 30
  4581.4  803.61  4613.4  801.31  4651.7   789.6    4657  790.07  4676.6   785.4
    4682  785.84  4706.9  776.94  4720.2   776.2  4730.9  773.46  4737.1   770.6
  4767.4  766.98  4773.6  765.03  4792.3  762.49  4805.7  761.34  4822.6  763.87
  4859.1  764.37  4913.4  760.46  4923.1  758.32  4955.2   758.5  4977.5  756.05
    4978  755.55    4997  756.05  4998.8  757.66  5018.9  760.43  5026.6  763.95
  5031.8  764.16  5049.8  770.43  5067.9  773.88    5122  777.99  5214.7  781.96
#Mann= 3 ,-1 , 0
  4581.4     .12       0  4977.5     .05       0    4997     .12       0
Bank Sta=4977.5,4997
XS Rating Curve= 0 ,0
Exp/Cntr=0.3,0.1

Type RM Length L Ch R = 1 ,1890    ,438,438,438
BEGIN DESCRIPTION:
A19245
END DESCRIPTION:
XS GIS Cut Line= 3
      2236047.25     13865367.52      2234666.51     13865390.25
      2233643.77     13865481.16
#Sta/Elev= 30
    3678  982.61  3681.6  982.61  3700.3  962.39  3720.3  949.02  3820.3  894.96
  3900.3  848.54  3920.3  846.99  3980.3  821.96  4040.3  807.04  4130.3  790.63
  4192.8  786.03  4330.3  775.51  4669.7  772.06  4781.1  767.33  4870.4  753.18
  4920.4  757.04  4950.4  756.12  4980.7  749.55  4981.2  749.05  5000.2  749.55
  5018.5  756.91  5030.4  765.89  5039.6  768.33  5077.1  770.33  5222.7  777.06
  5542.6  791.43  5662.8  805.73  5847.6  821.02  6014.2  849.11  6085.7  855.84
#Mann= 10 ,-1 , 0
    3678     .12       0  4192.8    .035       0  4669.7     .07       0
  4781.1     .12       0  4980.7     .05       0  5000.2     .12       0
  5018.5      .1       0  5077.1     .12       0  5222.7    .035       0
  5542.6     .12       0
Bank Sta=4980.7,5000.2
XS Rating Curve= 0 ,0
Exp/Cntr=0.3,0.1

Type RM Length L Ch R = 1 ,1452    ,516,516,516
BEGIN DESCRIPTION:
A19244
END DESCRIPTION:
XS GIS Cut Line= 2
      2236115.42     13865003.87      2233649.71     13865100.46
#Sta/Elev= 30
  3808.9  927.44  3884.8  905.19  3964.9   868.8  3969.9  874.78  3999.5  872.23
  4059.5  853.18  4083.8  850.63  4109.5     843  4189.6  802.97  4237.2  789.01
  4378.5   777.7  4816.4  768.57  4950.2  767.82  4970.9  764.24  5010.4  742.31
  5010.9  741.81    5030  742.31  5050.3  751.97  5060.3  752.78  5080.3  745.06
  5130.3  747.19  5168.3  758.46  5239.1  784.97  5323.7  793.15  5365.8  794.16
  5560.8     797  5657.7   799.5  5840.5   805.5  6081.1  817.09  6276.5  837.27
#Mann= 15 ,-1 , 0
  3808.9    .035       0  3884.8     .12       0  4083.8    .035       0
  4237.2     .12       0  4378.5    .035       0  4816.4     .07       0
  4970.9      .1       0  5010.4     .05       0    5030      .1       0
  5168.3    .035       0  5323.7     .12       0  5365.8     .07       0
  5560.8     .12       0  5657.7    .035       0  5840.5     .12       0
Bank Sta=5010.4,5030
XS Rating Curve= 0 ,0
Exp/Cntr=0.3,0.1
