--- LITTLE CREEK.prj (project) ---

Proj Title=LITTLE CREEK Base Level Engineering
Current Plan=p01
Default Exp/Contr=0.3,0.1
English Units
Geom File=g01
Flow File=f01
Plan File=p01
Y Axis Title=Elevation
X Axis Title(PF)=Main Channel Distance
X Axis Title(XS)=Station
BEGIN DESCRIPTION:
LITTLE CREEK
END DESCRIPTION:
DSS Export Rating Curves= 0
DSS Export Rating Curve Sorted= 0
DSS Export Volume Flow Curves= 0
DXF OffsetX= 0
DXF OffsetY= 0
DXF ScaleX= 1
DXF ScaleY= 10

--- LITTLE CREEK.p01 (plan) ---

Plan Title=Multiple Run
Short Identifier=Multiple
Geom File=g01
Flow File=f01
Subcritical Flow
K Sum by GR= 0
Std Step Tol= 0.01
Critical Tol= 0.01
Num of Std Step Trials= 20
Max Error Tol= 0.3
Flow Tol Ratio= 0.001
Split Flow NTrial= 30
Split Flow Tol= 0.02
Split Flow Ratio= 0.02
Log Output Level= 0
Friction Slope Method= 1
Unsteady Friction Slope Method= 2
Unsteady Bridges Friction Slope Method= 1
Parabolic Critical Depth
Global Vel Dist=  1 , 1 , 1
Global Log Level= 0
CheckData=True
Encroach Param= -1, 0, 0, 0
BEGIN DESCRIPTION:
Multiple Run
END DESCRIPTION:

--- LITTLE CREEK.f01 (steady flow) ---

Flow Title=Multiple
Number of Profiles=7
Profile Names=10-year,25-year,50-year,1pct_min,100-year,1pct_plu,500-year
River Rch & RM= LITTLE CREEK,Reach-1,38194
     512     824    1107     722    1441    2875    2416
River Rch & RM= LITTLE CREEK,Reach-1,36102
    1137    1914    2645    1768    3528    7039    6225
River Rch & RM= LITTLE CREEK,Reach-1,28419
    1255    2115    2925    1956    3903    7787    6890
River Rch & RM= LITTLE CREEK,Reach-1,23393
    1650    2818    3933    2651    5290   10555    9492
River Rch & RM= LITTLE CREEK,Reach-1,21984
    2204    3786    5303    3582    7147   14261   12880
River Rch & RM= LITTLE CREEK,Reach-1,16027
    2188    3751    5247    3539    7060   14087   12685
River Rch & RM= LITTLE CREEK,Reach-1,14654
    2277    3898    5445    3666    7314   14594   13095
River Rch & RM= LITTLE CREEK,Reach-1,9787
    2231    3796    5280    3538    7060   14086   12526
Boundary for River Rch & Prof#=LITTLE CREEK,Reach-1,1
Up Type=0
Dn Type=3
Dn Slope=0.005
Boundary for River Rch & Prof#=LITTLE CREEK,Reach-1,2
Up Type=0
Dn Type=3
Dn Slope=0.005
Boundary for River Rch & Prof#=LITTLE CREEK,Reach-1,3
Up Type=0
Dn Type=3
Dn Slope=0.005
Boundary for River Rch & Prof#=LITTLE CREEK,Reach-1,4
Up Type=0
Dn Type=3
Dn Slope=0.005
Boundary for River Rch & Prof#=LITTLE CREEK,Reach-1,5
Up Type=0
Dn Type=3
Dn Slope=0.005
Boundary for River Rch & Prof#=LITTLE CREEK,Reach-1,6
Up Type=0
Dn Type=3
Dn Slope=0.005
Boundary for River Rch & Prof#=LITTLE CREEK,Reach-1,7
Up Type=0
Dn Type=3
Dn Slope=0.005

--- LITTLE CREEK.g01 (geometry) ---

Geom Title=Existing Conditions

River Reach=LITTLE CREEK,Reach-1
Reach XY= 30
      2313175.00     13795825.00      2312480.83     13795077.30
      2312525.00     13794475.00      2311732.60     13793178.34
      2311919.92     13792122.69      2311411.20     13792061.81
      2310425.87     13790914.67      2310674.41     13788085.62
      2309925.98     13787235.26      2310817.17     13786781.18
      2311174.81     13786109.65      2310951.12     13785648.06
      2311619.54     13785527.47      2311867.21     13784125.10
      2311119.16     13782022.71      2309826.19     13780714.50
      2310721.54     13778376.49      2310077.31     13777680.82
      2309083.13     13777431.08      2309367.16     13775921.77
      2308427.14     13775169.03      2308738.52     13773961.59
      2309521.56     13773823.78      2309180.52     13772922.02
      2309925.69     13772695.07      2309627.74     13772230.34
      2309030.52     13772227.44      2308979.97     13771572.42
      2309472.74     13771380.94      2308575.00     13770325.00

Type RM Length L Ch R = 1,38194,362,362,362
BEGIN DESCRIPTION:
A19679
END DESCRIPTION:
XS GIS Cut Line= 2
      2313435.39     13795531.77      2312672.99     13796066.45
#Sta/Elev= 30
  4638.4  643.64  4663.3  644.29  4780.6  641.00  4791.8  640.35  4821.4  639.65
  4863.3  639.20  4928.6  637.54  4949.6  637.38  4970.5  636.57  4979.2  635.69
  4991.1  635.12  4991.3  634.62  4994.8  634.62  4995.1  635.12  5029.7  635.63
  5050.7  638.85  5056.8  640.31  5065.5  641.40  5071.6  641.55  5078.6  641.04
  5092.5  638.88  5102.2  637.93  5177.2  638.79  5334.9  640.66  5386.6  641.15
  5464.6  641.70  5517.9  641.65  5524.0  641.93  5538.8  641.18  5569.6  642.61
#Mann=9,-1,0
  4638.4   0.035       0  4780.6    0.07       0  4991.1   0.035       0
  4995.1    0.07       0  5102.2    0.07       0  5177.2   0.035       0
  5334.9   0.045       0  5386.6   0.035       0  5464.6    0.07       0
Bank Sta=4991.1,4995.1
Exp/Cntr=0.3,0.1

Type RM Length L Ch R = 1,37832,223,223,223
BEGIN DESCRIPTION:
LITTLE CREEK 68.0
END DESCRIPTION:
XS GIS Cut Line= 3
      2313325.03     13795425.00      2312925.00     13795475.00
      2312524.97     13796075.04
#Sta/Elev= 30
  4591.4  642.09  4629.2  640.87  4672.1  640.06  4742.6  637.32  4833.3  635.56
  4917.4  633.28  4956.7  632.41  4990.0  631.21  4990.3  630.71  4993.8  630.71
  4994.0  631.21  4997.5  631.21  5002.1  632.32  5030.6  631.94  5203.4  634.51
  5326.6  637.25  5347.6  637.07  5362.6  637.54  5368.6  637.19  5377.6  637.43
  5383.6  636.69  5397.3  637.50  5398.7  637.62  5404.7  636.08  5419.7  637.16
  5455.8  638.65  5506.8  639.54  5527.9  639.49  5639.3  640.84  5715.7  641.88
#Mann=6,-1,0
  4591.4   0.035       0  4917.4   0.045       0  4990.0   0.045       0
  4994.0   0.045       0  5397.3    0.07       0  5639.3   0.045       0
Bank Sta=4990,4994
Exp/Cntr=0.3,0.1

Type RM Length L Ch R = 1,37609,248,248,248
BEGIN DESCRIPTION:
A19678
END DESCRIPTION:
XS GIS Cut Line= 4
      2313178.03     13795221.49      2312788.52     13795297.41
      2312729.11     13795360.12      2312524.89     13795841.03
#Sta/Elev= 30
  4574.1  637.70  4620.8  637.30  4665.5  636.46  4727.4  634.94  4801.3  632.48
  4832.3  631.90  4930.4  628.63  4964.3  628.02  4985.8  628.38  4991.1  627.10
  4991.3  626.60  4994.8  626.60  4995.1  627.10  5000.0  627.60  5007.2  629.39
  5028.3  629.36  5076.1  630.14  5127.1  629.83  5173.0  630.76  5178.6  630.84
  5193.0  630.22  5238.0  632.49  5256.2  633.12  5261.7  632.82  5277.1  633.23
  5285.3  633.01  5382.7  635.12  5414.5  635.24  5449.3  635.98  5579.8  637.88
#Mann=11,-1,0
  4574.1   0.035       0  4665.5    0.05       0  4727.4   0.035       0
  4991.1   0.035       0  4995.1   0.035       0  5076.1   0.045       0
  5173.0    0.07       0  5178.6   0.035       0  5277.1   0.045       0
  5382.7    0.07       0  5449.3   0.045       0
Bank Sta=4991.1,4995.1
Exp/Cntr=0.3,0.1

Type RM Length L Ch R = 1,37361,424,424,424
BEGIN DESCRIPTION:
LITTLE CREEK 67.0
END DESCRIPTION:
XS GIS Cut Line= 3
      2313024.97     13795175.00      2312575.00     13795175.00
      2312525.00     13795624.96
#Sta/Elev= 30
  4549.7  634.58  4552.2  634.58  4659.7  631.50  4686.2  630.91  4749.7  628.85
  4759.7  628.63  4839.7  625.93  4869.7  625.29  4884.2  625.40  4939.7  625.81
  4949.7  625.59  4959.7  625.09  4969.7  624.48  4977.7  623.62  4977.9  623.12
  4981.4  623.12  4981.7  623.62  4997.2  625.17  5002.2  625.17  5009.7  625.56
  5080.2  627.41  5090.1  627.99  5100.3  628.59  5110.3  628.87  5130.5  628.89
  5180.8  629.59  5211.0  630.68  5221.0  630.77  5231.1  630.20  5452.4  634.14
#Mann=6,-1,0
  4549.7    0.05       0  4686.2   0.035       0  4884.2    0.07       0
  4977.7    0.07       0  4981.7    0.07       0  5090.1   0.045       0
Bank Sta=4977.7,4981.7
Exp/Cntr=0.3,0.1

Type RM Length L Ch R = 1,36937,367,367,367
BEGIN DESCRIPTION:
LITTLE CREEK 66.0
END DESCRIPTION:
XS GIS Cut Line= 3
      2312975.02     13795125.01      2312375.00     13794825.00
      2311475.03     13794875.00
#Sta/Elev= 30
  4329.0  633.05  4381.8  631.83  4532.4  627.24  4605.7  624.24  4700.8  621.90
  4739.9  622.28  4784.6  620.86  4983.9  619.46  4984.1  618.96  4987.6  618.96
  4987.9  619.46  5094.3  619.70  5120.0  619.63  5130.0  620.45  5150.1  623.31
  5180.1  620.69  5210.2  619.93  5240.2  621.89  5260.2  624.14  5272.8  624.59
  5280.3  624.64  5300.3  622.87  5320.3  621.99  5422.6  622.23  5590.8  624.18
  5610.8  625.03  5721.0  627.17  5759.9  628.37  5813.6  629.22  5901.2  631.74
#Mann=8,-1,0
  4329.0    0.05       0  4381.8   0.035       0  4532.4    0.05       0
  4983.9    0.05       0  4987.9    0.05       0  5094.3    0.07       0
  5422.6    0.05       0  5759.9   0.035       0
Bank Sta=4983.9,4987.9
Exp/Cntr=0.3,0.1

Type RM Length L Ch R = 1,36570,468,468,468
BEGIN DESCRIPTION:
A19677
END DESCRIPTION:
XS GIS Cut Line= 3
      2312913.97     13794812.25      2312412.25     13794488.77
      2311739.48     13794633.88
#Sta/Elev= 30
  4480.2  627.40  4520.9  626.27  4572.4  625.60  4645.0  623.21  4681.2  622.63
  4727.8  621.12  4728.7  621.10  4752.6  620.68  4802.1  618.97  4843.7  618.78
  4883.5  618.67  4917.4  618.12  4990.6  617.31  5017.9  616.77  5018.2  616.27
  5021.7  616.27  5021.9  616.77  5056.2  617.10  5076.0  617.00  5086.3  617.36
  5112.4  617.51  5146.0  617.98  5197.1  619.65  5340.9  620.62  5505.7  621.74
  5608.1  622.43  5637.0  623.27  5657.5  623.07  5688.1  623.39  5765.4  624.80
#Mann=10,-1,0
  4480.2   0.035       0  4727.8    0.07       0  4728.7    0.05       0
  4843.7   0.035       0  4917.4    0.07       0  5017.9    0.07       0
  5021.9    0.07       0  5112.4    0.05       0  5340.9    0.07       0
  5505.7    0.05       0
Bank Sta=5017.9,5021.9
Exp/Cntr=0.3,0.1

Type RM Length L Ch R = 1,36102,477,477,477
BEGIN DESCRIPTION:
LITTLE CREEK 65.0
END DESCRIPTION:
XS GIS Cut Line= 3
      2312975.03     13794074.99      2312375.00     13794175.00
      2311775.02     13794574.99
#Sta/Elev= 30
  4380.1  629.00  4805.9  617.76  4894.6  614.61  4951.8  614.23  4991.4  613.89
  4995.9  612.74  5017.0  614.08  5032.0  613.92  5038.0  613.66  5045.0  611.84
  5045.2  611.34  5048.7  611.34  5049.0  611.84  5053.0  613.15  5060.5  613.92
  5161.2  616.86  5176.2  617.19  5191.2  618.34  5197.2  620.26  5218.3  620.66
  5248.3  620.61  5263.3  620.06  5269.3  619.25  5299.4  619.07  5326.4  619.82
  5371.5  619.81  5557.8  621.51  5587.8  622.55  5608.9  622.19  5709.5  623.83
#Mann=6,-1,0
  4380.1   0.035       0  4951.8    0.07       0  5045.0    0.07       0
  5049.0    0.07       0  5161.2   0.035       0  5371.5    0.05       0
Bank Sta=5045,5049
Exp/Cntr=0.3,0.1

Type RM Length L Ch R = 1,35625,440,440,440
BEGIN DESCRIPTION:
LITTLE CREEK 64.0
END DESCRIPTION:
XS GIS Cut Line= 3
      2312774.97     13793525.01      2312175.00     13793775.00
      2311574.98     13794225.02
#Sta/Elev= 30
  4344.8  627.55  4492.2  623.25  4521.8  622.24  4600.2  619.89  4708.3  616.97
  4802.5  614.26  4820.9  613.26  4843.1  613.58  4901.6  611.45  4927.1  610.95
  4950.9  611.20  4980.1  610.57  4985.6  608.61  5000.1  608.45  5000.3  607.95
  5003.8  607.95  5004.1  608.45  5008.3  609.87  5031.2  609.79  5087.5  610.77
  5152.4  610.46  5187.5  610.65  5202.1  610.01  5216.6  609.97  5402.1  613.82
  5552.1  619.14  5687.5  623.34  5702.1  623.97  5722.9  625.68  5744.8  626.49
#Mann=9,-1,0
  4344.8   0.045       0  4492.2    0.07       0  4521.8   0.045       0
  4600.2    0.07       0  4708.3   0.035       0  4901.6    0.07       0
  5000.1    0.07       0  5004.1    0.07       0  5152.4   0.035       0
Bank Sta=5000.1,5004.1
Exp/Cntr=0.3,0.1

Type RM Length L Ch R = 1,35185,449,449,449
BEGIN DESCRIPTION:
LITTLE CREEK 63.0
END DESCRIPTION:
XS GIS Cut Line= 3
      2312274.97     13793425.01      2312125.00     13793475.00
      2311525.01     13793974.99
#Sta/Elev= 30
  4837.9  614.49  4865.0  613.89  4901.1  611.72  4911.7  612.58  4943.3  611.77
  4974.9  609.64  4993.3  606.87  4999.2  606.87  5003.1  604.42  5007.7  603.93
  5007.9  603.43  5011.4  603.43  5011.7  603.93  5017.5  605.69  5052.6  607.40
  5087.8  608.17  5095.6  607.83  5102.1  605.57  5109.9  607.83  5116.4  606.17
  5124.2  607.65  5152.2  608.87  5223.1  609.11  5251.8  608.53  5406.7  610.38
  5529.0  613.68  5658.9  619.37  5746.5  622.64  5751.8  622.83  5777.0  623.71
#Mann=8,-1,0
  4837.9   0.035       0  4865.0    0.07       0  5007.7    0.07       0
  5011.7    0.07       0  5406.7   0.035       0  5658.9    0.07       0
  5746.5   0.035       0  5751.8    0.07       0
Bank Sta=5007.7,5011.7
Exp/Cntr=0.3,0.1

Type RM Length L Ch R = 1,34736,468,468,468
BEGIN DESCRIPTION:
LITTLE CREEK 62.0
END DESCRIPTION:
XS GIS Cut Line= 3
      2312374.99     13793075.00      2311775.00     13793225.00
      2311525.00     13793275.00
#Sta/Elev= 30
  4381.1  618.68  4481.6  615.26  4537.4  613.85  4566.8  613.15  4646.5  610.68
  4710.9  609.60  4721.2  609.84  4729.0  607.18  4741.9  605.32  4811.4  604.72
  4816.6  604.92  4824.3  606.12  4834.6  609.11  4844.9  611.17  4857.8  611.51
  4865.6  611.24  4875.9  609.80  4886.2  606.45  4893.9  604.71  4940.3  604.91
  4989.2  603.73  4995.0  602.78  4995.2  602.28  4998.7  602.28  4999.0  602.78
  5030.1  605.18  5101.5  609.72  5152.5  610.50  5183.1  611.79  5254.5  613.84
#Mann=5,-1,0
  4381.1    0.07       0  4537.4   0.035       0  4566.8    0.07       0
  4995.0    0.07       0  4999.0    0.07       0
Bank Sta=4995,4999
Exp/Cntr=0.3,0.1

Type RM Length L Ch R = 1,34268,449,449,449
BEGIN DESCRIPTION:
LITTLE CREEK 61.0
END DESCRIPTION:
XS GIS Cut Line= 3
      2312075.05     13792875.01      2311775.00     13792825.00
      2311574.99     13792975.01
#Sta/Elev= 30
  4694.8  609.93  4722.7  608.69  4727.8  608.69  4803.0  605.64  4836.8  604.17
  4844.4  603.65  4849.4  603.63  4857.1  603.10  4905.2  601.39  4910.3  601.65
  4938.2  600.97  4958.4  600.87  4971.1  600.54  4978.7  600.05  4986.8  599.11
  4987.1  598.61  4990.6  598.61  4990.8  599.11  4996.5  600.34  5002.1  600.34
  5006.3  602.67  5012.5  601.75  5020.9  602.90  5062.5  603.36  5091.7  604.43
  5106.3  605.32  5141.7  606.87  5191.7  608.26  5206.3  608.91  5249.0  610.24
#Mann=4,-1,0
  4694.8   0.045       0  4803.0    0.07       0  4986.8    0.07       0
  4990.8    0.07       0
Bank Sta=4986.8,4990.8
Exp/Cntr=0.3,0.1

Type RM Length L Ch R = 1,33819,473,473,473
BEGIN DESCRIPTION:
LITTLE CREEK 60.0
END DESCRIPTION:
XS GIS Cut Line= 3
      2312075.02     13792425.00      2311825.00     13792425.00
      2311475.03     13792674.98
#Sta/Elev= 30
  4749.4  607.96  4801.1  605.73  4829.4  604.52  4839.4  604.25  4899.4  601.01
  4926.4  599.73  4939.4  599.17  4959.4  598.88  4969.4  598.34  4987.4  596.50
  4987.7  596.00  4991.2  596.00  4991.4  596.50  4996.9  597.45  5002.5  597.45
  5006.8  598.07  5021.5  598.57  5036.3  598.79  5047.7  599.24  5092.8  600.70
  5102.4  600.82  5122.3  601.52  5128.5  601.57  5134.6  602.05  5149.3  602.26
  5164.1  602.24  5171.3  602.45  5418.6  607.37  5427.7  607.69  5429.5  607.69
#Mann=10,-1,0
  4749.4   0.035       0  4801.1    0.07       0  4926.4    0.16       0
  4987.4    0.07       0  4991.4    0.16       0  5047.7    0.07       0
  5102.4    0.16       0  5171.3   0.035       0  5418.6   0.045       0
  5427.7    0.07       0
Bank Sta=4987.4,4991.4
Exp/Cntr=0.3,0.1

Type RM Length L Ch R = 1,33346,482,482,482
BEGIN DESCRIPTION:
LITTLE CREEK 59.0
END DESCRIPTION:
XS GIS Cut Line= 3
      2311925.04     13791974.98      2311825.00     13792025.00
      2311274.98     13792575.02
#Sta/Elev= 30
  4883.9  605.46  4886.7  605.46  4892.3  605.11  4897.9  604.97  4906.3  604.56
  4914.3  603.89  4920.3  603.52  4932.9  602.02  4942.6  600.87  4951.0  599.43
  4965.0  597.55  4973.4  596.68  4981.8  596.13  4993.0  595.72  5022.0  595.42
  5022.3  594.92  5025.8  594.92  5026.0  595.42  5038.2  595.96  5052.3  596.31
  5090.1  596.02  5123.0  595.77  5165.5  596.04  5225.3  597.41  5278.6  599.34
  5321.7  599.78  5335.2  599.75  5420.0  600.91  5770.0  608.78  5773.6  608.78
#Mann=8,-1,0
  4883.9   0.045       0  4914.3    0.07       0  4932.9    0.16       0
  5022.0    0.07       0  5026.0    0.16       0  5090.1    0.07       0
  5225.3   0.035       0  5321.7   0.045       0
Bank Sta=5022,5026
Exp/Cntr=0.3,0.1

Type RM Length L Ch R = 1,32864,464,464,464
BEGIN DESCRIPTION:
LITTLE CREEK 58.0
END DESCRIPTION:
XS GIS Cut Line= 3
      2311674.98     13791825.01      2311375.00     13792025.00
      2311375.00     13792174.97
#Sta/Elev= 30
  4642.9  601.25  4701.5  599.30  4743.5  597.31  4764.6  596.68  4773.6  596.59
  4830.7  594.52  4851.7  594.11  4902.8  592.48  4944.8  593.43  4959.9  593.36
  4967.4  593.53  4974.9  592.46  4980.9  592.17  4989.9  590.56  4993.9  590.52
  4994.2  590.02  4997.7  590.02  4997.9  590.52  5000.4  590.79  5005.9  590.79
  5013.4  592.33  5023.4  591.81  5033.4  593.10  5043.4  595.09  5053.4  596.66
  5058.9  597.20  5073.4  598.39  5083.4  598.96  5123.4  600.23  5153.4  600.66
#Mann=4,-1,0
  4642.9    0.07       0  4993.9    0.07       0  4997.9    0.07       0
  5058.9   0.035       0
Bank Sta=4993.9,4997.9
Exp/Cntr=0.3,0.1

Type RM Length L Ch R = 1,32400,423,423,423
BEGIN DESCRIPTION:
LITTLE CREEK 57.0
END DESCRIPTION:
XS GIS Cut Line= 3
      2311425.04     13791625.00      2311275.00     13791625.00
      2311125.02     13791824.97
#Sta/Elev= 30
  4850.6  597.24  4853.1  597.24  4920.6  594.77  4930.6  594.25  4950.6  592.97
  4960.6  592.55  4970.6  592.01  4980.6  590.67  4990.6  588.98  4996.1  586.29
  4996.4  585.79  4999.9  585.79  5000.1  586.29  5003.8  586.29  5007.9  586.67
  5014.2  587.03  5022.5  587.75  5028.8  587.96  5057.9  590.03  5087.1  591.15
  5107.9  592.15  5114.2  592.56  5122.5  592.77  5128.8  593.11  5176.4  594.63
  5187.1  594.98  5222.5  596.38  5243.3  596.89  5247.5  597.13  5250.6  597.13
#Mann=4,-1,0
  4850.6    0.07       0  4996.1    0.07       0  5000.1    0.07       0
  5176.4   0.035       0
Bank Sta=4996.1,5000.1
Exp/Cntr=0.3,0.1

Type RM Length L Ch R = 1,31977,414,414,414
BEGIN DESCRIPTION:
LITTLE CREEK 56.0
END DESCRIPTION:
XS GIS Cut Line= 3
      2311174.98     13791275.01      2311025.00     13791325.00
      2310924.99     13791475.02
#Sta/Elev= 30
  4846.5  593.16  4888.6  592.16  4893.4  591.90  4899.2  591.58  4920.3  590.89
  4930.8  590.02  4962.4  588.30  4973.0  586.45  4983.5  583.41  4992.1  582.79
  4992.3  582.29  4995.8  582.29  4996.1  582.79  4998.2  583.30  5002.0  584.21
  5007.6  584.21  5012.1  586.22  5018.1  586.55  5027.1  586.77  5033.1  587.56
  5048.2  588.54  5070.8  589.39  5084.2  590.06  5105.3  590.70  5120.3  591.50
  5171.4  593.07  5177.4  593.31  5179.0  593.48  5181.9  593.78  5184.9  593.78
#Mann=7,-1,0
  4846.5   0.035       0  4893.4    0.16       0  4992.1    0.07       0
  4996.1    0.16       0  4998.2    0.07       0  5070.8    0.16       0
  5179.0    0.07       0
Bank Sta=4992.1,4996.1
Exp/Cntr=0.3,0.1

Type RM Length L Ch R = 1,31563,405,405,405
BEGIN DESCRIPTION:
LITTLE CREEK 55.0
END DESCRIPTION:
XS GIS Cut Line= 3
      2311025.00     13790975.00      2310775.00     13791025.00
      2310674.99     13791325.02
#Sta/Elev= 30
  4741.1  590.94  4812.5  589.58  4822.7  589.10  4868.2  587.87  4945.1  586.69
  4965.5  586.83  4985.9  586.16  4993.5  583.31  4998.7  583.31  5004.6  580.79
  5004.8  580.29  5008.3  580.29  5008.6  580.79  5017.1  581.33  5027.7  583.72
  5038.2  584.79  5048.8  585.62  5052.0  585.62  5059.3  585.63  5066.8  585.43
  5080.4  585.07  5090.9  585.08  5133.1  585.79  5164.7  586.12  5185.8  586.73
  5196.3  587.13  5228.0  588.83  5249.0  590.31  5270.1  591.30  5312.3  592.58
#Mann=6,-1,0
  4741.1    0.05       0  4868.2    0.07       0  5004.6    0.07       0
  5008.6    0.07       0  5052.0    0.16       0  5066.8    0.07       0
Bank Sta=5004.6,5008.6
Exp/Cntr=0.3,0.1

Type RM Length L Ch R = 1,31158,444,444,444
BEGIN DESCRIPTION:
LITTLE CREEK 54.0
END DESCRIPTION:
XS GIS Cut Line= 3
      2310974.97     13790775.01      2310425.00     13790925.00
      2310324.98     13791025.02
#Sta/Elev= 30
  4433.6  590.32  4456.0  590.09  4530.3  588.65  4651.2  585.60  4666.9  585.40
  4758.3  583.99  4792.9  582.89  4819.8  582.92  4827.4  582.98  4837.8  583.49
  4872.4  583.86  4906.9  583.10  4931.1  583.20  4951.8  582.99  4962.2  583.16
  4972.6  581.96  4981.2  580.58  4984.4  579.47  4984.6  578.97  4988.1  578.97
  4988.4  579.47  4993.3  580.84  5001.1  583.92  5007.2  583.92  5017.8  586.41
  5031.9  587.52  5065.2  588.12  5088.5  588.40  5108.1  589.00  5145.1  589.80
#Mann=7,-1,0
  4433.6    0.05       0  4666.9    0.07       0  4819.8    0.16       0
  4984.4    0.07       0  4988.4    0.16       0  5065.2    0.07       0
  5108.1   0.035       0
Bank Sta=4984.4,4988.4
Exp/Cntr=0.3,0.1

Type RM Length L Ch R = 1,30714,453,453,453
BEGIN DESCRIPTION:
LITTLE CREEK 53.0
END DESCRIPTION:
XS GIS Cut Line= 3
      2311074.96     13790724.99      2310375.00     13790525.00
      2310025.03     13790874.97
#Sta/Elev= 30
  4280.2  591.74  4409.1  589.64  4554.5  587.01  4612.0  585.44  4627.3  585.08
  4661.1  583.50  4700.1  583.36  4713.6  582.90  4733.9  582.25  4739.1  582.42
  4806.7  581.14  4873.0  581.34  4925.0  580.76  4957.5  581.13  4989.3  580.66
  4989.5  580.16  4993.0  580.16  4993.3  580.66  4997.8  581.38  5005.6  581.72
  5022.3  581.85  5135.4  581.01  5177.9  581.21  5255.7  583.45  5262.7  585.02
  5291.0  584.90  5339.7  586.41  5390.0  587.96  5474.9  591.83  5503.1  592.45
#Mann=7,-1,0
  4280.2   0.035       0  4409.1    0.05       0  4612.0    0.07       0
  4713.6    0.16       0  4989.3    0.07       0  4993.3    0.16       0
  5339.7   0.035       0
Bank Sta=4989.3,4993.3
Exp/Cntr=0.3,0.1

Type RM Length L Ch R = 1,30261,487,487,487
BEGIN DESCRIPTION:
LITTLE CREEK 52.0
END DESCRIPTION:
XS GIS Cut Line= 3
      2311074.97     13790524.98      2310525.00     13790125.00
      2308724.97     13791125.02
#Sta/Elev= 30
  4320.0  590.54  4687.0  584.32  4877.5  581.57  4906.9  580.40  4957.1  576.23
  4992.7  575.93  4994.9  575.12  4995.2  574.62  4998.9  575.12  5035.5  576.88
  5065.7  580.55  5116.7  583.89  5125.9  583.48  5132.7  580.46  5205.9  580.59
  5331.8  579.92  5382.1  582.18  5411.9  580.13  5441.6  581.64  5448.3  580.78
  5469.1  580.02  5582.3  580.65  5837.4  588.44  6080.5  587.68  6088.6  587.62
  6189.0  587.28  6355.1  587.55  6662.0  586.04  6772.2  585.91  7059.2  584.81
#Mann=13,-1,0
  4320.0   0.035       0  4687.0    0.07       0  4994.9    0.07       0
  4998.9    0.07       0  5065.7    0.16       0  5205.9   0.033       0
  5448.3    0.16       0  6080.5    0.07       0  6088.6    0.16       0
  6189.0    0.07       0  6355.1   0.045       0  6662.0    0.07       0
  6772.2   0.045       0
Bank Sta=4994.9,4998.9
Exp/Cntr=0.3,0.1

Type RM Length L Ch R = 1,29774,432,432,432
BEGIN DESCRIPTION:
LITTLE CREEK 51.0
END DESCRIPTION:
XS GIS Cut Line= 3
      2311024.96     13790124.97      2310425.00     13789675.00
      2309774.99     13790325.01
#Sta/Elev= 30
  4250.0  585.95  4513.5  581.62  4571.8  582.15  4636.4  580.78  4692.7  580.91
  4750.0  579.87  4807.2  577.00  4857.2  575.39  4863.5  575.95  4886.4  573.12
  4928.5  572.68  4978.1  572.98  4992.7  570.98  4994.8  569.99  4995.0  569.49
  4998.6  569.49  4998.9  569.99  5014.1  571.11  5042.4  571.56  5084.8  574.59
  5113.1  575.32  5141.4  574.72  5155.5  573.72  5169.7  575.74  5212.1  577.70
  5410.1  580.02  5678.8  580.86  5749.5  581.80  5820.2  584.43  5919.2  586.28
#Mann=4,-1,0
  4250.0    0.07       0  4928.5    0.16       0  4994.8    0.07       0
  4998.9    0.16       0
Bank Sta=4994.8,4998.9
Exp/Cntr=0.3,0.1

Type RM Length L Ch R = 1,29342,457,457,457
BEGIN DESCRIPTION:
LITTLE CREEK 50.0
END DESCRIPTION:
XS GIS Cut Line= 3
      2311024.98     13789774.99      2310475.00     13789275.00
      2308674.98     13789275.00
#Sta/Elev= 30
  4274.8  582.30  4430.5  580.59  4685.3  573.67  4819.8  572.03  4954.2  571.29
  4961.7  567.81  4968.4  568.89  4980.6  567.23  4980.8  566.73  4984.4  566.73
  4984.7  567.23  4990.0  568.15  4996.8  567.38  5004.2  568.04  5011.0  567.60
  5014.7  568.95  5053.2  569.36  5208.1  570.56  5338.1  569.73  5378.1  568.99
  5398.1  567.90  5418.1  570.78  5485.1  573.54  5508.1  574.78  5608.1  577.43
  5682.0  578.44  5828.1  580.45  6296.2  581.67  6324.9  581.52  6818.1  582.37
#Mann=8,-1,0
  4274.8    0.07       0  4980.6    0.07       0  4984.7    0.07       0
  5053.2    0.16       0  5485.1    0.07       0  5682.0   0.045       0
  6296.2   0.035       0  6324.9   0.045       0
Bank Sta=4980.6,4984.7
Exp/Cntr=0.3,0.1

Type RM Length L Ch R = 1,28885,466,466,466
BEGIN DESCRIPTION:
LITTLE CREEK 49.0
END DESCRIPTION:
XS GIS Cut Line= 3
      2311025.02     13789575.02      2310475.00     13788925.00
      2309725.01     13789125.00
#Sta/Elev= 30
  4143.3  579.88  4214.2  579.15  4384.5  574.57  4526.2  571.92  4774.5  569.64
  4881.1  569.71  4923.9  569.18  4938.2  568.33  4941.3  568.96  4944.8  569.67
  4981.1  568.86  4987.7  567.61  4997.4  567.65  5005.2  565.05  5014.6  564.41
  5015.1  563.91  5019.8  563.91  5020.2  564.41  5025.8  566.17  5057.5  566.75
  5067.2  566.26  5108.6  566.84  5132.6  565.76  5150.0  567.38  5167.5  570.17
  5172.7  569.88  5191.4  571.29  5471.2  575.46  5593.1  578.21  5771.0  579.63
#Mann=5,-1,0
  4143.3    0.07       0  4941.3    0.16       0  5014.6    0.07       0
  5020.2    0.16       0  5471.2   0.045       0
Bank Sta=5014.6,5020.2
Exp/Cntr=0.3,0.1

Type RM Length L Ch R = 1,28419,449,449,449
BEGIN DESCRIPTION:
LITTLE CREEK 48.0
END DESCRIPTION:
XS GIS Cut Line= 3
      2311525.02     13788575.00      2310725.00     13788575.00
      2310125.00     13788525.00
#Sta/Elev= 30
  4195.7  587.48  4356.7  581.08  4370.6  580.57  4549.6  574.47  4635.7  570.63
  4685.7  569.07  4755.7  568.67  4875.7  566.54  4885.7  566.63  4905.7  570.00
  4915.7  570.39  4935.7  567.82  4965.7  568.08  4975.7  565.83  4982.6  561.63
  4983.1  561.13  4988.3  561.13  4988.8  561.63  4998.2  561.88  5005.8  563.07
  5015.8  563.66  5045.9  563.89  5076.0  565.32  5146.2  566.24  5178.9  565.41
  5226.5  567.35  5298.4  567.92  5419.7  571.39  5535.1  575.57  5597.8  576.89
#Mann=7,-1,0
  4195.7    0.07       0  4356.7    0.16       0  4370.6    0.07       0
  4549.6    0.16       0  4982.6    0.07       0  4988.8    0.16       0
  5298.4    0.07       0
Bank Sta=4982.6,4988.8
Exp/Cntr=0.3,0.1

Type RM Length L Ch R = 1,27970,448,448,448
BEGIN DESCRIPTION:
LITTLE CREEK 47.0
END DESCRIPTION:
XS GIS Cut Line= 3
      2311425.03     13787924.99      2310625.00     13788225.00
      2310175.00     13788275.00
#Sta/Elev= 30
  4140.2  583.78  4185.6  582.12  4342.9  574.51  4450.0  568.49  4503.4  567.02
  4643.1  565.09  4662.7  564.27  4668.0  565.71  4674.2  564.69  4684.9  564.00
  4692.9  564.89  4698.3  564.58  4717.0  566.21  4759.7  563.09  4802.4  562.98
  4899.4  564.12  4984.8  563.78  5024.8  562.51  5031.7  560.12  5032.2  559.62
  5037.5  559.62  5038.0  560.12  5044.9  560.17  5055.0  563.78  5065.1  565.32
  5095.2  566.07  5125.4  567.51  5161.3  567.83  5306.5  572.98  5447.4  576.12
#Mann=5,-1,0
  4140.2    0.07       0  4342.9    0.16       0  5031.7    0.07       0
  5038.0    0.16       0  5161.3    0.07       0
Bank Sta=5031.7,5038
Exp/Cntr=0.3,0.1

Type RM Length L Ch R = 1,27522,384,384,384
BEGIN DESCRIPTION:
LITTLE CREEK 46.0
END DESCRIPTION:
XS GIS Cut Line= 3
      2311025.02     13787574.99      2310475.00     13787875.00
      2310225.02     13788174.98
#Sta/Elev= 30
  4373.5  575.92  4431.0  573.84  4485.1  572.51  4572.4  569.00  4610.4  568.58
  4695.5  566.44  4713.8  565.93  4719.5  565.97  4726.6  566.57  4735.7  566.40
  4749.4  565.34  4801.2  564.72  4851.9  563.64  4888.5  563.64  4932.1  562.68
  4942.6  563.00  4964.4  562.31  4986.3  560.41  4988.8  559.85  4989.3  559.35
  4994.7  559.35  4995.2  559.85  5007.2  560.19  5042.3  563.87  5056.6  564.37
  5117.7  565.24  5198.5  568.28  5220.7  569.64  5312.4  572.91  5390.5  574.78
#Mann=5,-1,0
  4373.5    0.07       0  4695.5    0.16       0  4988.8    0.07       0
  4995.2    0.16       0  5117.7    0.07       0
Bank Sta=4988.8,4995.2
Exp/Cntr=0.3,0.1

Type RM Length L Ch R = 1,27138,524,524,524
BEGIN DESCRIPTION:
A19676
END DESCRIPTION:
XS GIS Cut Line= 3
      2310960.01     13787541.79      2310292.12     13787518.96
      2309726.97     13788186.86
#Sta/Elev= 30
  4139.5  574.67  4190.8  572.87  4274.6  570.98  4413.4  568.61  4463.3  568.04
  4554.8  566.57  4624.8  566.12  4704.8  566.93  4810.1  565.50  4885.1  563.17
  4951.8  562.59  4966.1  561.73  4980.4  559.79  4986.9  560.02  4991.5  559.65
  4992.0  559.15  4997.4  559.15  4997.9  559.65  5009.0  561.43  5023.3  561.96
  5044.1  562.27  5101.3  564.20  5136.4  564.77  5150.7  565.85  5185.8  566.68
  5359.8  572.79  5440.5  574.78  5505.6  575.52  5571.7  575.56  5682.7  575.82
#Mann=9,-1,0
  4139.5    0.07       0  4413.4    0.16       0  4463.3    0.07       0
  4885.1    0.16       0  4991.5    0.07       0  4997.9    0.16       0
  5359.8   0.035       0  5440.5    0.07       0  5571.7   0.035       0
Bank Sta=4991.5,4997.9
Exp/Cntr=0.3,0.1

Type RM Length L Ch R = 1,26614,448,448,448
BEGIN DESCRIPTION:
LITTLE CREEK 45.0
END DESCRIPTION:
XS GIS Cut Line= 3
      2311125.05     13787525.01      2309925.00     13787325.00
      2309525.00     13787625.00
#Sta/Elev= 30
  3783.3  578.54  3811.2  577.74  3877.1  577.22  4054.5  572.14  4358.7  566.90
  4432.2  566.07  4503.1  566.43  4555.0  565.93  4602.0  565.16  4675.5  562.96
  4756.6  562.07  4776.9  560.93  4850.4  560.31  4939.1  560.86  4972.0  559.46
  4979.6  560.53  4989.8  560.59  5003.0  560.27  5007.2  558.34  5010.2  558.29
  5010.7  557.79  5016.2  557.79  5016.7  558.29  5021.8  559.47  5071.8  564.06
  5139.3  565.57  5207.2  568.60  5242.6  569.23  5323.9  572.12  5499.9  573.91
#Mann=6,-1,0
  3783.3    0.07       0  4555.0   0.035       0  5010.2   0.035       0
  5016.7   0.035       0  5139.3    0.16       0  5323.9   0.035       0
Bank Sta=5010.2,5016.7
Exp/Cntr=0.3,0.1

Type RM Length L Ch R = 1,26166,489,489,489
BEGIN DESCRIPTION:
LITTLE CREEK 44.0
END DESCRIPTION:
XS GIS Cut Line= 3
      2310774.99     13787374.99      2310225.00     13787075.00
      2309925.00     13786925.00
#Sta/Elev= 30
  4367.4  571.05  4381.2  570.93  4419.1  569.53  4447.1  569.46  4545.9  567.69
  4566.3  567.32  4631.8  564.37  4647.9  564.80  4668.4  564.46  4778.9  560.63
  4876.7  559.36  4926.0  557.65  4996.7  557.20  5016.2  556.29  5021.4  555.01
  5021.9  554.51  5027.4  554.51  5027.9  555.01  5030.2  556.64  5063.3  559.75
  5074.9  561.13  5091.7  562.36  5097.3  563.21  5107.7  563.41  5142.0  564.70
  5181.2  565.37  5217.5  567.51  5239.9  567.42  5270.0  568.71  5329.3  570.48
#Mann=8,-1,0
  4367.4    0.07       0  4545.9   0.035       0  4668.4    0.07       0
  5021.4    0.07       0  5027.9    0.07       0  5063.3    0.16       0
  5107.7    0.07       0  5270.0   0.045       0
Bank Sta=5021.4,5027.9
Exp/Cntr=0.3,0.1

Type RM Length L Ch R = 1,25677,476,476,476
BEGIN DESCRIPTION:
LITTLE CREEK 43.0
END DESCRIPTION:
XS GIS Cut Line= 3
      2310774.99     13787124.99      2310675.00     13786975.00
      2310324.98     13786724.99
#Sta/Elev= 30
  4815.2  569.30  4816.3  569.30  4915.8  564.52  4981.9  559.26  4992.5  557.23
  4998.5  557.23  5005.4  555.52  5020.4  553.21  5020.9  552.71  5027.0  553.21
  5059.4  555.41  5124.0  556.85  5195.8  560.15  5216.7  564.97  5231.4  567.05
  5246.2  567.95  5253.5  566.93  5260.9  564.49  5267.1  564.11  5275.7  560.72
  5281.8  561.66  5290.4  558.83  5311.3  558.64  5317.4  561.32  5326.0  561.37
  5332.2  564.18  5346.9  564.78  5353.1  565.98  5388.7  567.69  5425.6  568.10
#Mann=7,-1,0
  4815.2    0.07       0  4816.3    0.16       0  5005.4   0.035       0
  5020.4    0.07       0  5027.0   0.035       0  5124.0    0.16       0
  5231.4    0.07       0
Bank Sta=5020.4,5027
Exp/Cntr=0.3,0.1

Type RM Length L Ch R = 1,25201,416,416,416
BEGIN DESCRIPTION:
LITTLE CREEK 42.0
END DESCRIPTION:
XS GIS Cut Line= 3
      2311125.01     13786775.01      2310875.00     13786575.00
      2310525.02     13786525.00
#Sta/Elev= 30
  4679.8  569.28  4800.7  563.76  4815.1  562.57  4843.9  558.83  4850.3  558.65
  4858.3  557.64  4864.7  558.76  4871.9  557.34  4885.5  557.71  4901.8  556.83
  4907.9  556.40  4914.3  556.87  4922.3  556.08  4928.7  556.58  4957.5  554.46
  4978.4  553.80  4986.4  552.87  4992.8  553.04  4993.5  552.32  4994.0  551.82
  4999.6  551.82  5000.1  552.32  5010.1  553.18  5020.2  552.95  5050.5  554.87
  5121.2  556.82  5197.6  560.42  5296.7  563.70  5333.3  566.71  5353.5  566.67
#Mann=6,-1,0
  4679.8    0.07       0  4901.8    0.16       0  4993.5    0.07       0
  5000.1    0.16       0  5197.6   0.035       0  5296.7    0.07       0
Bank Sta=4993.5,5000.1
Exp/Cntr=0.3,0.1

Type RM Length L Ch R = 1,24785,464,464,464
BEGIN DESCRIPTION:
LITTLE CREEK 41.0
END DESCRIPTION:
XS GIS Cut Line= 3
      2311325.01     13786575.02      2311075.00     13786225.00
      2310525.01     13786275.00
#Sta/Elev= 30
  4575.2  568.89  4653.9  566.05  4719.0  562.51  4775.5  559.02  4805.0  557.90
  4811.2  557.43  4882.4  555.43  4926.7  554.65  4946.9  553.58  4956.2  553.01
  4968.5  551.72  4977.1  551.29  4979.9  550.11  4980.4  549.61  4986.0  549.61
  4986.5  550.11  4991.8  551.13  5002.3  551.93  5065.6  553.07  5095.7  554.21
  5226.2  556.63  5326.7  560.02  5356.8  561.49  5394.1  562.80  5417.0  563.64
  5493.3  565.40  5507.4  566.04  5527.5  567.97  5537.5  568.20  5557.6  567.32
#Mann=6,-1,0
  4575.2    0.07       0  4946.9    0.16       0  4979.9    0.07       0
  4986.5    0.16       0  5394.1   0.035       0  5493.3    0.07       0
Bank Sta=4979.9,4986.5
Exp/Cntr=0.3,0.1

Type RM Length L Ch R = 1,24321,248,248,248
BEGIN DESCRIPTION:
LITTLE CREEK 40.0
END DESCRIPTION:
XS GIS Cut Line= 3
      2311424.97     13786224.97      2311025.00     13785875.00
      2310624.98     13786225.02
#Sta/Elev= 30
  4472.0  564.68  4656.6  560.28  4741.0  559.56  4748.6  557.81  4755.3  558.27
  4762.9  554.65  4769.5  554.82  4777.1  553.39  4783.7  557.22  4798.0  553.79
  4804.6  558.62  4864.0  556.84  4925.2  554.02  4932.8  552.72  4939.4  553.76
  4953.6  553.63  4961.2  552.21  4967.9  552.99  4975.5  551.19  4982.1  552.58
  4989.7  550.28  4996.3  551.64  4996.8  549.29  4997.3  548.79  5003.5  549.29
  5074.2  552.27  5286.8  554.71  5372.2  559.20  5447.9  561.56  5535.0  564.44
#Mann=5,-1,0
  4472.0    0.07       0  4864.0    0.16       0  4996.8    0.07       0
  5003.5    0.16       0  5447.9   0.035       0
Bank Sta=4996.8,5003.5
Exp/Cntr=0.3,0.1

Type RM Length L Ch R = 1,24073,232,232,232
BEGIN DESCRIPTION:
A19675
END DESCRIPTION:
XS GIS Cut Line= 3
      2311376.77     13786143.20      2311011.40     13785686.49
      2310183.66     13785526.65
#Sta/Elev= 30
  4333.6  563.16  4678.9  556.20  4803.7  552.24  4867.7  551.00  4965.7  551.90
  4992.9  548.94  4993.4  548.44  4999.6  548.94  5016.7  550.15  5026.8  551.93
  5037.0  552.38  5112.2  551.31  5223.1  552.16  5352.7  551.48  5371.3  549.95
  5388.8  552.93  5413.9  555.05  5434.2  554.03  5444.4  554.81  5454.6  557.70
  5464.8  558.65  5485.2  554.04  5495.3  553.01  5525.9  552.51  5546.3  554.29
  5566.6  557.36  5601.2  558.61  5687.4  562.55  5729.6  563.25  5761.5  564.85
#Mann=7,-1,0
  4333.6    0.07       0  4678.9    0.16       0  4992.9    0.07       0
  4999.6    0.16       0  5223.1   0.035       0  5388.8    0.16       0
  5601.2    0.07       0
Bank Sta=4992.9,4999.6
Exp/Cntr=0.3,0.1

Type RM Length L Ch R = 1,23841,448,448,448
BEGIN DESCRIPTION:
LITTLE CREEK 39.0
END DESCRIPTION:
XS GIS Cut Line= 3
      2311424.98     13786174.96      2311125.00     13785575.00
      2310524.98     13784924.98
#Sta/Elev= 30
  4329.1  564.35  4700.8  556.73  4840.6  551.00  5007.0  548.75  5056.3  550.39
  5325.6  548.77  5367.6  550.34  5389.2  548.73  5396.0  549.21  5403.3  547.89
  5449.3  547.31  5449.8  546.81  5456.0  547.31  5486.7  548.02  5530.6  548.23
  5537.7  549.50  5544.5  548.60  5551.9  550.25  5587.1  549.51  5629.6  550.87
  5672.1  554.67  5679.5  556.50  5700.5  558.42  5714.6  561.62  5742.4  562.17
  5785.5  562.51  5805.5  564.05  5828.0  564.37  5834.9  563.07  5884.5  564.46
#Mann=7,-1,0
  4329.1    0.07       0  4840.6    0.16       0  5449.3    0.07       0
  5456.0    0.16       0  5486.7   0.035       0  5742.4    0.16       0
  5805.5    0.07       0
Bank Sta=5449.3,5456
Exp/Cntr=0.3,0.1

Type RM Length L Ch R = 1,23393,473,473,473
BEGIN DESCRIPTION:
LITTLE CREEK 38.0
END DESCRIPTION:
XS GIS Cut Line= 3
      2311425.01     13786024.97      2311525.00     13785625.00
      2310975.02     13784875.03
#Sta/Elev= 30
  4584.1  561.15  4725.8  556.57  4731.0  555.90  4790.2  555.37  4808.3  553.22
  4813.4  551.98  4837.0  553.24  4883.0  554.83  4913.9  552.94  4965.5  551.40
  4973.2  549.62  4978.3  549.33  4993.8  546.12  4996.4  546.12  4999.5  544.92
  5000.0  544.42  5007.5  544.42  5008.0  544.92  5018.4  545.78  5068.5  546.55
  5118.7  546.15  5254.5  548.28  5396.6  548.88  5607.7  553.38  5618.1  553.60
  5626.6  554.96  5641.2  555.31  5726.9  555.91  5797.9  558.57  5926.4  560.67
#Mann=5,-1,0
  4584.1    0.07       0  4837.0    0.16       0  4999.5    0.07       0
  5008.0    0.16       0  5607.7   0.045       0
Bank Sta=4999.5,5008
Exp/Cntr=0.3,0.1

Type RM Length L Ch R = 1,22920,558,558,558
BEGIN DESCRIPTION:
LITTLE CREEK 37.0
END DESCRIPTION:
XS GIS Cut Line= 3
      2312075.01     13785575.01      2311725.00     13785225.00
      2311225.00     13784825.00
#Sta/Elev= 30
  4500.7  559.37  4543.1  558.29  4619.8  554.88  4868.4  548.61  4882.6  547.72
  4889.6  547.66  4896.7  546.92  4925.0  545.24  4939.1  545.06  4967.4  545.79
  4981.5  545.59  4992.2  544.01  4995.7  544.01  4998.2  543.38  4998.7  542.88
  5007.0  542.88  5007.5  543.38  5009.3  544.56  5017.3  545.63  5046.1  546.29
  5091.2  546.14  5159.8  547.63  5244.6  548.48  5372.7  551.03  5436.7  552.80
  5443.9  553.15  5451.1  554.71  5465.5  555.31  5572.0  557.71  5636.0  558.68
#Mann=5,-1,0
  4500.7   0.035       0  4619.8    0.16       0  4998.2    0.07       0
  5007.5    0.16       0  5091.2   0.045       0
Bank Sta=4998.2,5007.5
Exp/Cntr=0.3,0.1

Type RM Length L Ch R = 1,22362,378,378,378
BEGIN DESCRIPTION:
A19674
END DESCRIPTION:
XS GIS Cut Line= 3
      2312141.72     13785555.22      2311924.78     13784744.57
      2311218.46     13784647.74
#Sta/Elev= 30
  4068.9  558.98  4115.0  558.30  4229.9  554.70  4264.8  554.54  4304.8  552.97
  4322.8  552.75  4419.8  550.86  4425.0  551.45  4431.4  550.70  4459.8  549.63
  4574.8  547.90  4648.8  547.92  4809.9  546.90  4910.5  546.99  4942.5  546.07
  4973.9  543.70  4974.4  543.20  4982.7  543.20  4983.2  543.70  5039.1  545.94
  5079.4  545.35  5138.5  546.30  5163.9  546.65  5170.3  548.26  5180.4  548.13
  5210.7  549.49  5291.4  551.13  5402.4  554.72  5563.9  557.16  5621.0  558.57
#Mann=5,-1,0
  4068.9   0.035       0  4322.8    0.16       0  4973.9    0.07       0
  4983.2    0.16       0  5138.5   0.045       0
Bank Sta=4973.9,4983.2
Exp/Cntr=0.3,0.1

Type RM Length L Ch R = 1,21984,440,440,440
BEGIN DESCRIPTION:
LITTLE CREEK 36.0
END DESCRIPTION:
XS GIS Cut Line= 3
      2312275.02     13784224.99      2311875.00     13784375.00
      2311225.00     13784575.00
#Sta/Elev= 30
  4572.8  563.02  4648.5  559.63  4703.7  556.54  4728.6  554.73  4767.9  552.76
  4783.8  551.92  4819.4  551.07  4838.9  549.91  4861.2  549.41  4929.7  546.09
  4954.6  545.58  4968.0  545.77  4984.0  543.16  4984.5  542.66  4996.0  542.66
  4996.5  543.16  5010.5  543.34  5016.4  544.79  5021.6  544.93  5031.4  546.25
  5041.9  547.12  5054.3  547.54  5073.3  546.91  5125.6  546.66  5155.5  547.30
  5209.3  548.20  5353.8  552.65  5391.7  552.92  5522.5  556.25  5680.1  558.62
#Mann=5,-1,0
  4572.8   0.045       0  4767.9    0.16       0  4984.0    0.07       0
  4996.5    0.16       0  5155.5   0.045       0
Bank Sta=4984,4996.5
Exp/Cntr=0.3,0.1

Type RM Length L Ch R = 1,21544,447,447,447
BEGIN DESCRIPTION:
LITTLE CREEK 35.0
END DESCRIPTION:
XS GIS Cut Line= 3
      2312124.99     13783875.00      2311825.00     13783975.00
      2311124.98     13784425.01
#Sta/Elev= 30
  4683.8  560.05  4694.3  559.86  4799.7  553.10  4853.7  550.90  4884.1  550.03
  4894.6  548.53  4905.1  548.35  4926.2  546.55  4968.4  545.25  4983.2  544.16
  4983.7  543.66  4995.3  543.66  4995.8  544.16  5007.6  545.16  5013.6  544.63
  5043.9  545.72  5143.3  544.98  5253.7  547.24  5319.3  548.49  5464.9  552.95
  5528.0  553.30  5564.4  554.61  5579.6  554.63  5600.7  553.71  5606.6  554.74
  5611.5  554.64  5637.0  555.14  5643.0  554.25  5737.1  557.73  5832.2  559.55
#Mann=8,-1,0
  4683.8   0.035       0  4853.7    0.16       0  4983.2    0.07       0
  4995.8    0.16       0  5143.3   0.035       0  5253.7   0.045       0
  5464.9   0.035       0  5611.5   0.045       0
Bank Sta=4983.2,4995.8
Exp/Cntr=0.3,0.1

Type RM Length L Ch R = 1,21097,485,485,485
BEGIN DESCRIPTION:
LITTLE CREEK 34.0
END DESCRIPTION:
XS GIS Cut Line= 3
      2312025.01     13783625.00      2311675.00     13783575.00
      2311124.97     13784075.02
#Sta/Elev= 30
  4645.9  557.90  4676.2  557.06  4794.0  550.86  4898.4  547.65  4949.0  543.64
  4969.2  543.19  4973.0  541.33  4973.5  540.83  4985.1  540.83  4985.6  541.33
  4989.4  542.62  4996.9  543.91  5029.6  544.35  5055.9  545.00  5077.5  544.74
  5254.6  546.41  5268.7  546.81  5275.5  547.78  5289.7  548.65  5318.1  549.22
  5332.3  549.01  5346.4  549.75  5354.8  549.46  5360.6  549.44  5367.4  548.31
  5389.0  548.62  5403.2  549.61  5496.6  550.79  5558.6  551.62  5742.8  556.17
#Mann=7,-1,0
  4645.9    0.05       0  4794.0    0.07       0  4973.0    0.07       0
  4985.6    0.07       0  5029.6    0.05       0  5354.8   0.035       0
  5496.6   0.045       0
Bank Sta=4973,4985.6
Exp/Cntr=0.3,0.1

Type RM Length L Ch R = 1,20612,459,459,459
BEGIN DESCRIPTION:
LITTLE CREEK 33.0
END DESCRIPTION:
XS GIS Cut Line= 3
      2312375.00     13782525.00      2311575.00     13783125.00
      2310775.01     13784324.99
#Sta/Elev= 30
  3995.7  562.20  4374.4  560.41  4503.0  557.84  4798.9  544.98  4827.6  544.68
  4853.0  543.67  4923.8  544.47  4967.3  541.80  4967.8  541.30  4980.3  541.80
  4992.6  543.40  5090.3  542.77  5249.9  545.00  5356.3  545.17  5622.2  552.89
  5739.3  553.77  5766.4  554.97  5781.4  555.02  5796.4  553.38  5813.6  553.95
  5817.5  554.04  5825.0  551.05  5832.5  553.56  5847.5  554.49  5929.6  554.88
  5955.7  554.60  6069.8  557.77  6303.6  560.41  6337.1  560.89  6437.9  562.03
#Mann=11,-1,0
  3995.7    0.05       0  4374.4    0.07       0  4798.9   0.035       0
  4827.6    0.07       0  4967.3    0.07       0  4980.3    0.07       0
  5249.9    0.05       0  5813.6   0.035       0  5929.6   0.045       0
  6303.6   0.035       0  6337.1   0.045       0
Bank Sta=4967.3,4980.3
Exp/Cntr=0.3,0.1

Type RM Length L Ch R = 1,20153,439,439,439
BEGIN DESCRIPTION:
LITTLE CREEK 32.0
END DESCRIPTION:
XS GIS Cut Line= 3
      2312024.98     13782675.00      2311425.00     13782775.00
      2310425.01     13783474.99
#Sta/Elev= 30
  4396.1  560.13  4446.8  559.74  4497.5  559.14  4547.1  557.36  4647.4  553.19
  4780.9  546.87  4848.1  544.18  4923.3  542.13  4963.8  542.58  4976.5  541.59
  4977.4  539.79  4977.9  539.29  4990.7  539.79  4994.2  541.98  5001.8  542.67
  5154.8  544.06  5203.1  545.30  5235.0  546.05  5291.1  549.10  5378.0  551.34
  5419.8  551.30  5615.7  554.48  5800.8  556.19  5895.4  557.93  6009.2  558.07
  6017.5  556.52  6030.1  556.35  6038.5  557.99  6053.7  558.86  6225.0  560.01
#Mann=12,-1,0
  4396.1    0.07       0  4446.8    0.05       0  4547.1   0.035       0
  4647.4    0.07       0  4780.9    0.16       0  4848.1    0.05       0
  4977.4    0.05       0  4990.7    0.05       0  5203.1    0.07       0
  5291.1    0.05       0  5615.7    0.07       0  6038.5   0.045       0
Bank Sta=4977.4,4990.7
Exp/Cntr=0.3,0.1

Type RM Length L Ch R = 1,19714,429,429,429
BEGIN DESCRIPTION:
LITTLE CREEK 31.0
END DESCRIPTION:
XS GIS Cut Line= 3
      2311774.98     13782225.01      2311225.00     13782425.00
      2310424.98     13783325.02
#Sta/Elev= 30
  4419.3  559.46  4526.4  558.21  4582.2  556.70  4674.9  550.38  4760.4  546.50
  4837.9  544.15  4918.9  542.08  4983.2  541.63  4987.9  540.40  4988.4  539.90
  5001.2  540.40  5001.9  541.63  5032.5  542.43  5061.0  541.99  5146.3  543.39
  5393.8  550.01  5667.4  553.49  5727.0  554.95  5827.6  555.75  5868.8  556.65
  5932.3  556.14  5939.8  556.67  5945.5  555.38  5975.0  554.86  5981.6  557.56
  6010.1  557.32  6052.7  559.18  6060.2  558.31  6074.5  558.32  6208.7  559.29
#Mann=9,-1,0
  4419.3    0.05       0  4674.9    0.07       0  4837.9    0.16       0
  4918.9    0.07       0  4987.9    0.07       0  5001.2    0.07       0
  5667.4    0.05       0  5827.6    0.07       0  5945.5   0.045       0
Bank Sta=4987.9,5001.2
Exp/Cntr=0.3,0.1

Type RM Length L Ch R = 1,19285,468,468,468
BEGIN DESCRIPTION:
LITTLE CREEK 30.0
END DESCRIPTION:
XS GIS Cut Line= 3
      2311725.04     13782125.01      2311125.00     13782025.00
      2310024.97     13782825.02
#Sta/Elev= 30
  4387.2  559.11  4416.5  559.06  4497.7  558.20  4569.7  557.20  4658.4  552.33
  4846.0  544.63  4884.0  541.81  4914.4  541.43  4934.7  542.68  4962.6  540.33
  4967.6  541.03  4968.5  539.54  4969.0  539.04  4981.9  539.54  5017.5  541.59
  5082.1  540.58  5109.5  541.98  5189.1  543.13  5195.3  544.33  5224.7  544.65
  5239.3  543.28  5245.5  544.52  5587.4  550.57  5603.3  551.10  5611.8  548.64
  5638.9  549.93  5647.4  551.73  5689.1  552.58  6197.6  558.44  6355.7  559.38
#Mann=6,-1,0
  4387.2    0.07       0  4416.5   0.045       0  4497.7    0.07       0
  4968.5    0.07       0  4981.9    0.07       0  5587.4   0.045       0
Bank Sta=4968.5,4981.9
Exp/Cntr=0.3,0.1

Type RM Length L Ch R = 1,18817,470,470,470
BEGIN DESCRIPTION:
LITTLE CREEK 29.0
END DESCRIPTION:
XS GIS Cut Line= 3
      2312025.01     13781175.00      2310825.00     13781675.00
      2309825.02     13782674.98
#Sta/Elev= 30
  3703.9  561.09  3794.4  559.81  3855.6  558.62  3872.4  559.17  3888.1  557.66
  3925.5  558.24  4034.1  555.20  4142.1  550.93  4181.0  550.15  4223.9  547.96
  4238.5  549.24  4264.9  547.42  4331.6  546.99  4440.0  546.62  4469.3  544.93
  4537.5  544.30  4798.1  540.86  4898.1  540.89  4898.2  540.89  4989.3  540.05
  4994.3  539.12  4994.8  538.62  5008.1  539.12  5102.9  543.19  5682.7  551.75
  5711.0  551.05  5739.3  553.49  5746.4  552.65  5852.4  553.35  6418.1  559.81
#Mann=12,-1,0
  3703.9   0.045       0  3794.4   0.035       0  4034.1    0.16       0
  4142.1    0.07       0  4181.0    0.16       0  4264.9    0.07       0
  4331.6    0.16       0  4537.5   0.045       0  4898.1   0.035       0
  4898.2    0.07       0  4994.3    0.07       0  5008.1   0.045       0
Bank Sta=4994.3,5008.1
Exp/Cntr=0.3,0.1

Type RM Length L Ch R = 1,18347,468,468,468
BEGIN DESCRIPTION:
LITTLE CREEK 28.0
END DESCRIPTION:
XS GIS Cut Line= 3
      2311625.01     13780675.00      2310625.00     13781275.00
      2309724.97     13782275.03
#Sta/Elev= 30
  3829.7  558.34  3864.7  558.84  3888.0  556.18  3895.8  557.48  3923.0  557.29
  3946.3  554.47  3991.3  552.56  4129.0  551.21  4193.2  549.46  4279.3  549.63
  4478.9  550.46  4696.6  544.31  4840.5  542.14  4980.8  540.43  4999.3  539.91
  5002.8  536.39  5003.3  535.89  5016.6  536.39  5031.4  538.86  5068.3  540.79
  5314.7  542.17  5767.6  548.03  5796.0  547.45  5916.4  550.74  5959.0  550.27
  6008.3  552.32  6157.0  554.83  6199.6  553.68  6242.2  555.94  6341.3  557.39
#Mann=8,-1,0
  3829.7   0.035       0  3991.3    0.07       0  4279.3   0.045       0
  4840.5   0.035       0  4980.8    0.05       0  5002.8    0.05       0
  5016.6    0.05       0  5068.3   0.045       0
Bank Sta=5002.8,5016.6
Exp/Cntr=0.3,0.1

Type RM Length L Ch R = 1,17879,467,467,467
BEGIN DESCRIPTION:
LITTLE CREEK 27.0
END DESCRIPTION:
XS GIS Cut Line= 3
      2311425.03     13780474.99      2310225.00     13781075.00
      2309624.98     13782075.03
#Sta/Elev= 30
  3654.1  556.71  3698.9  555.61  3868.0  549.76  3964.3  547.02  4439.3  547.75
  4552.2  548.46  4713.5  548.77  4830.9  543.05  4870.0  542.74  4907.0  540.22
  4920.3  539.52  4937.1  540.78  4942.7  539.40  4951.0  540.11  4959.4  539.06
  4981.8  541.46  4987.4  538.59  4998.7  538.33  5012.1  535.28  5012.6  534.78
  5026.0  535.28  5049.2  538.09  5061.9  539.53  5162.0  540.08  5274.8  541.55
  5718.8  546.06  5878.2  549.04  5979.3  552.78  6010.4  551.92  6162.0  555.66
#Mann=12,-1,0
  3654.1   0.035       0  3698.9   0.045       0  3868.0    0.07       0
  3964.3   0.045       0  4439.3   0.035       0  4552.2    0.05       0
  4907.0    0.07       0  5012.1    0.07       0  5026.0    0.07       0
  5049.2    0.05       0  5162.0   0.035       0  5274.8   0.045       0
Bank Sta=5012.1,5026
Exp/Cntr=0.3,0.1

Type RM Length L Ch R = 1,17412,450,450,450
BEGIN DESCRIPTION:
LITTLE CREEK 26.0
END DESCRIPTION:
XS GIS Cut Line= 3
      2311525.01     13780375.00      2309875.00     13780825.00
      2308887.83     13781210.93
#Sta/Elev= 30
  3294.3  560.10  3377.2  559.52  3466.1  556.27  3613.1  552.62  3634.9  551.81
  3733.1  547.72  3885.0  544.80  3961.0  543.21  4193.8  544.86  4328.1  547.48
  4341.4  547.48  4444.8  548.66  4838.7  538.99  4937.2  538.58  4994.2  538.34
  5002.0  536.06  5012.4  535.43  5012.9  534.93  5026.5  535.43  5040.5  538.65
  5147.4  539.44  5296.4  540.20  5338.4  542.05  5498.5  546.81  5530.7  545.98
  5605.8  548.54  5646.7  547.84  5713.2  550.07  5760.7  549.71  6064.5  555.39
#Mann=15,-1,0
  3294.3   0.035       0  3466.1   0.045       0  3613.1    0.07       0
  3634.9   0.045       0  3885.0   0.035       0  3961.0   0.045       0
  4193.8    0.05       0  4328.1   0.035       0  4341.4    0.05       0
  4937.2    0.07       0  5012.4    0.07       0  5026.5    0.07       0
  5040.5    0.05       0  5147.4    0.07       0  5338.4   0.045       0
Bank Sta=5012.4,5026.5
Exp/Cntr=0.3,0.1
