HEC-RAS study LONG CREEK.prj: LONG CREEK Base Level Engineering

--- LONG CREEK.g01 (geometry) --- (continued)

Type RM Length L Ch R = 1 ,33183   ,441,441,441
BEGIN DESCRIPTION:
LONG CREEK 51.0
END DESCRIPTION:
XS GIS Cut Line= 3
      2255124.96     13775375.02        2256025.       13774775.
      2257224.99     13773875.01
#Sta/Elev= 30
  3906.8  618.73  4067.9  613.58  4172.1  608.48    4323  605.02  4368.1   605.1
  4398.1  603.18  4449.3  602.59  4533.3  599.86  4619.2   599.1  4680.2  598.79
  4772.2  597.08  4991.6   597.6  4995.8  593.61  5002.1   595.2  5010.4  592.99
    5024  592.97  5024.5  592.47  5038.4  592.97  5038.5  595.91  5045.8  598.61
    5122   599.2    5475  601.66  5562.5  602.26  5679.7  603.37  5749.9  604.02
  6066.6  607.79  6388.5  613.23  6402.1  614.71    6426  615.36  6488.5  615.87
#Mann= 16 ,-1 , 0
  3906.8    .045       0  4067.9     .07       0  4172.1    .045       0
    4323    .035       0  4449.3    .045       0  4619.2    .035       0
  4680.2     .07       0    5024     .05       0  5038.4     .07       0
    5122    .045       0    5475     .07       0  5562.5    .045       0
  5679.7    .035       0  5749.9    .045       0  6402.1     .07       0
    6426    .045       0
Bank Sta=5024,5038.4
XS Rating Curve= 0 ,0
Exp/Cntr=0.3,0.1

Type RM Length L Ch R = 1 ,32742   ,551,551,551
BEGIN DESCRIPTION:
LONG CREEK 50.0
END DESCRIPTION:
XS GIS Cut Line= 3
      2255424.98     13775575.01        2256025.       13775175.
      2257225.01     13773974.99
#Sta/Elev= 30
  4278.4  614.73    4301  615.25  4386.6  611.49  4430.2  611.14  4502.3  605.78
  4538.3  605.33  4589.4  602.46  4681.7  601.45  4697.6  601.93  4724.6  600.61
  4802.5  599.99  4810.9  599.78  4919.9  598.23    4977  596.49  4989.3  593.46
  4989.8  592.96  5003.8  593.46  5013.7  595.77  5098.5  596.38  5159.8  598.01
  5268.2  599.35  5339.5     599    5483  599.71  5697.3  601.01  5893.8  602.77
  5930.8  603.21  6057.2  604.83  6631.5  613.34  6661.2  613.81  6696.6  616.03
#Mann= 14 ,-1 , 0
  4278.4    .035       0  4681.7     .07       0  4802.5    .045       0
  4810.9     .07       0  4989.3     .05       0  5003.8     .07       0
  5159.8    .035       0  5339.5     .07       0    5483    .045       0
  5697.3     .07       0  5893.8    .045       0  5930.8    .035       0
  6057.2    .045       0  6631.5     .07       0
Bank Sta=4989.3,5003.8
XS Rating Curve= 0 ,0
Exp/Cntr=0.3,0.1

Type RM Length L Ch R = 1 ,32191   ,389,389,389
BEGIN DESCRIPTION:
A19804
END DESCRIPTION:
XS GIS Cut Line= 3
      2255829.83     13775955.78       2256420.1     13775532.18
      2257677.01     13775157.19
#Sta/Elev= 30
    4444   614.1  4490.8  614.07  4591.5  610.87  4627.1  611.79  4713.1  607.18
  4748.7  607.47  4784.3  604.21  4849.4   600.7  4899.7  600.07  4927.9  598.44
  4965.2  596.93  5015.2  594.78  5021.2  593.66  5021.7  593.16  5036.6  593.66
  5044.7  594.66  5086.4   596.4  5322.5  597.03  5421.9  599.17  5487.4  598.98
  5608.4   598.2    5611  598.25    5616  598.34    5687  599.54    5769  598.86
  5950.4  601.12  6135.7  605.17  6159.7   603.8  6198.3  605.33  6482.2  609.57
#Mann= 10 ,-1 , 0
    4444    .035       0  4927.9     .07       0  4965.2    .035       0
  5021.2    .035       0  5036.6    .035       0  5044.7     .07       0
  5487.4     .05       0  5608.4     .07       0    5611     .05       0
    5616    .035       0
Bank Sta=5021.2,5036.6
XS Rating Curve= 0 ,0
Exp/Cntr=0.3,0.1

Type RM Length L Ch R = 1 ,31802   ,469,469,469
BEGIN DESCRIPTION:
LONG CREEK 49.0
END DESCRIPTION:
XS GIS Cut Line= 3
      2256225.03     13776174.97        2256575.       13775875.
      2257800.99     13775192.49
#Sta/Elev= 30
  4538.8  612.71    4603  609.73    4631  610.44  4709.4  604.25  4736.9  604.22
  4787.4  599.29  4857.6   597.4  4881.4  595.69  4928.9   595.2  4964.1  593.74
  4992.6  594.39  5013.5  593.11  5021.7  590.91  5022.2  590.41  5037.2  590.91
  5045.5  595.11  5051.2  595.98  5179.9  596.79  5294.5  598.43  5335.4  598.66
  5576.7  600.53  5587.4  601.37  5594.9  600.61  5697.9  601.72  5800.9   604.1
  6042.5  605.01  6080.2  606.49  6137.4  607.32  6220.8   609.1  6402.9  611.05
#Mann= 9 ,-1 , 0
  4538.8    .035       0  4881.4     .07       0  5021.7     .05       0
  5037.2     .07       0  5179.9    .035       0  5294.5     .05       0
  5335.4    .035       0  5576.7     .05       0  6137.4    .035       0
Bank Sta=5021.7,5037.2
XS Rating Curve= 0 ,0
Exp/Cntr=0.3,0.1

Type RM Length L Ch R = 1 ,31333   ,419,419,419
BEGIN DESCRIPTION:
A19803
END DESCRIPTION:
XS GIS Cut Line= 3
      2256093.73     13776587.72       2256795.1     13776219.68
      2257885.35     13775309.97
#Sta/Elev= 30
  4301.1  620.31  4325.1  621.03  4445.3   615.3  4483.2  615.69  4562.3   611.9
    4594  612.57  4682.2  607.14  4709.9  608.04  4742.7  604.38  4814.5   601.3
  4845.2  598.68  4957.5  593.26  4968.9  591.83  4977.6  588.54  4978.1  588.04
  4993.1  588.54  5001.7  592.95  5007.4     594  5059.2  593.92  5133.2  596.27
    5182  597.85  5295.2  598.85  5475.3  597.45  5538.2  598.22  5685.7  599.22
  6012.4  604.68  6168.6  604.74  6307.5  609.05    6320  609.33  6513.1  611.37
#Mann= 9 ,-1 , 0
  4301.1    .035       0  4845.2     .07       0  4977.6     .05       0
  4993.1     .07       0  5133.2     .05       0  5475.3     .07       0
  5538.2     .05       0  6307.5     .07       0    6320    .035       0
Bank Sta=4977.6,4993.1
XS Rating Curve= 0 ,0
Exp/Cntr=0.3,0.1

Type RM Length L Ch R = 1 ,30914   ,826,826,826
BEGIN DESCRIPTION:
LONG CREEK 48.0
END DESCRIPTION:
XS GIS Cut Line= 3
      2256274.95     13776825.02        2256875.       13776625.
      2257940.92     13775428.02
#Sta/Elev= 30
  4371.7  618.13    4435     614  4466.6   613.8  4550.9  607.81  4614.2  604.84
  4688.1   603.6  4761.8  598.29  4867.2   594.2    4962  592.33  4972.6  589.81
  4975.4  587.45  4975.9  586.95  4990.9  587.45  4993.7  590.76  5001.6  593.47
  5039.7  593.75    5100  596.42  5174.4   598.5  5307.7  598.69  5356.4  598.83
  5436.1   599.3  5599.1  595.02  5673.6   595.7  5790.6  598.47  5864.5  598.58
  6130.1  603.28  6307.3  604.33  6441.8     608  6487.8  608.95    6607  610.75
#Mann= 12 ,-1 , 0
  4371.7    .035       0  4688.1     .07       0  4975.4     .05       0
  4990.9     .07       0    5100    .035       0  5307.7     .07       0
  5356.4    .035       0  5436.1     .05       0  5673.6     .07       0
  5864.5     .05       0  6441.8     .07       0  6487.8    .035       0
Bank Sta=4975.4,4990.9
XS Rating Curve= 0 ,0
Exp/Cntr=0.3,0.1

Type RM Length L Ch R = 1 ,30088   ,643,643,643
BEGIN DESCRIPTION:
LONG CREEK 47.0
END DESCRIPTION:
XS GIS Cut Line= 3
      2257149.27     13777698.82      2257302.04     13777226.62
      2257940.47     13775581.99
#Sta/Elev= 30
  4448.8  630.42    4812  617.18    4876  608.71  4902.7   603.9    4908  601.07
  4927.8  598.77    4940  594.56  4957.6  594.05  4970.4  589.55  4992.6  586.35
  4993.1  585.85  5008.4  586.35  5019.5  589.69  5043.4  591.28  5188.2  591.36
  5242.6  594.77    5248  593.09    5295  592.85  5700.5   593.4  5808.5  593.87
  6045.6  594.33    6179  596.04  6208.9  597.42  6214.3  599.55  6233.8  599.27
  6238.8  601.76  6354.2  600.32  6442.6  601.79  6607.3  606.18  6709.3  608.51
#Mann= 11 ,-1 , 0
  4448.8     .07       0  4927.8    .035       0  4992.6    .035       0
  5008.4    .035       0    5295     .07       0  5700.5     .05       0
  5808.5     .07       0  6233.8     .05       0  6354.2     .07       0
  6442.6     .05       0  6607.3     .07       0
Bank Sta=4992.6,5008.4
XS Rating Curve= 0 ,0
Exp/Cntr=0.3,0.1

Type RM Length L Ch R = 1 ,29445   ,550,550,550
BEGIN DESCRIPTION:
LONG CREEK 46.0
END DESCRIPTION:
XS GIS Cut Line= 3
      2257635.37     13777511.36      2257822.88     13777032.18
      2258121.25     13775588.86
#Sta/Elev= 30
  4376.4  617.85  4473.7  614.75  4551.7  608.99  4576.2  610.55    4606   606.3
  4660.3  606.96  4690.1  605.01  4705.4  600.64  4759.1   597.5  4834.2  598.47
  4898.3  588.04  4959.6  588.64  4992.5  585.02    4993  584.52  5008.3  585.02
    5031  589.57  5194.4  591.77  5255.7  589.23  5411.8  590.01  5511.7  590.89
  5611.6  594.16  5711.5  595.65  5772.2  596.57  5807.1  595.27  5878.6  600.14
  5911.3  598.16  6022.9  598.39  6111.1  602.73    6253  607.75  6364.8  609.69
#Mann= 13 ,-1 , 0
  4376.4    .035       0  4473.7     .07       0  4992.5     .05       0
  5008.3     .07       0  5411.8    .035       0  5511.7     .07       0
  5611.6     .05       0  5711.5     .07       0  5772.2     .05       0
  5911.3     .07       0  6022.9     .05       0  6111.1     .07       0
    6253    .035       0
Bank Sta=4992.5,5008.3
XS Rating Curve= 0 ,0
Exp/Cntr=0.3,0.1

Type RM Length L Ch R = 1 ,28895   ,642,642,642
BEGIN DESCRIPTION:
A19802
END DESCRIPTION:
XS GIS Cut Line= 3
      2257781.19     13777504.42       2258170.1     13777032.18
      2258274.27     13775830.75
#Sta/Elev= 30
  3891.5  614.69  3942.9  614.58  3963.8  613.18  4313.1  599.02  4413.7  596.17
  4593.2  592.06  4828.8  589.41  4881.9  588.07  4908.2  588.76  4966.2  586.56
  4972.2  588.07  4982.2  587.49  4984.2  584.44  4984.7  583.94  5000.3  584.44
  5022.4  588.78  5032.4  589.53  5105.3  587.72  5132.8  586.59    5183  594.33
  5197.4  593.89  5263.3   600.1  5309.7  600.64  5413.8  601.84  5474.1  601.47
  5484.1  600.21  5494.1   601.5  5504.2  600.56  5544.8  600.87  5709.2  604.32
#Mann= 11 ,-1 , 0
  3891.5    .035       0  3963.8     .07       0  4413.7    .035       0
  4593.2     .07       0  4828.8     .05       0  4908.2     .12       0
  4984.2     .05       0  5000.3     .12       0  5105.3     .07       0
  5309.7    .035       0  5544.8     .07       0
Bank Sta=4984.2,5000.3
XS Rating Curve= 0 ,0
Exp/Cntr=0.3,0.1

Type RM Length L Ch R = 1 ,28253   ,456,456,456
BEGIN DESCRIPTION:
LONG CREEK 45.0
END DESCRIPTION:
XS GIS Cut Line= 3
      2257524.97     13777825.03        2258725.       13776625.
      2258774.99     13776425.05
#Sta/Elev= 30
  3293.9  626.95  3407.1  622.83  3463.6  622.19  3590.9  617.86  3647.5  617.69
  3704.1   615.1  3810.3  612.63  4186.3  597.05  4368.7  591.15  4423.8  590.43
    4559   589.5    4694  589.21  4904.2  586.89  4976.9  586.92  4987.5  583.52
    5001   582.1  5001.5   581.6  5017.1   582.1  5021.9  585.55  5042.5  588.76
  5050.3  592.51  5055.4   597.2  5063.1  599.73  5083.8  597.78  5091.5  602.26
  5096.6  600.65  5104.4  603.51  5114.7  604.87  5149.4  605.45  5197.1   607.2
#Mann= 9 ,-1 , 0
  3293.9    .035       0  3810.3     .07       0  4186.3    .035       0
  4423.8     .07       0    4559     .05       0  4904.2     .12       0
    5001     .05       0  5017.1     .12       0  5149.4     .07       0
Bank Sta=5001,5017.1
XS Rating Curve= 0 ,0
Exp/Cntr=0.3,0.1

Type RM Length L Ch R = 1 ,27797   ,520,520,520
BEGIN DESCRIPTION:
LONG CREEK 44.0
END DESCRIPTION:
XS GIS Cut Line= 3
      2257875.02     13777624.99        2258875.       13777025.
      2259124.98     13776825.02
#Sta/Elev= 30
  3833.4  615.32  3891.7  615.26  3926.7  612.64    3950   612.8  4058.8  608.52
  4222.9  600.26  4271.9  597.81  4334.8  595.57  4427.7  590.77  4519.5     588
  4701.6  586.96  4906.3  585.15  4927.7   586.2  4964.6   586.2    4986  584.54
  4988.6  582.52  4989.1  582.02  5004.8  582.52  5021.2  586.42  5027.6  586.47
  5035.6   588.6    5042  588.57    5050  590.95  5056.4  589.67  5070.8  592.65
  5077.2  590.96  5111.9  595.15  5163.7  598.21  5251.4  600.91  5319.7  602.72
#Mann= 9 ,-1 , 0
  3833.4    .035       0  4222.9     .07       0  4271.9    .035       0
  4427.7     .07       0  4701.6     .05       0  4988.6     .05       0
  5004.8     .05       0  5111.9    .035       0  5251.4     .07       0
Bank Sta=4988.6,5004.8
XS Rating Curve= 0 ,0
Exp/Cntr=0.3,0.1

Type RM Length L Ch R = 1 ,27277   ,524,524,524
BEGIN DESCRIPTION:
A19801
END DESCRIPTION:
XS GIS Cut Line= 4
       2257885.4     13777934.94       2258482.6      13777504.4
      2258947.88     13777351.62      2259114.54     13776900.24
#Sta/Elev= 30
    4009  620.89  4036.9  620.94  4087.2  618.29  4137.6  618.31    4194   615.7
  4252.9  615.33  4294.6  612.73  4321.6  612.63  4353.5  612.03  4481.1  603.94
  4575.6  595.56  4609.7  593.89  4800.4   586.4  4863.5  585.99  4895.1  584.33
  4958.3  585.92  4978.9   582.6  4984.1  583.52  5007.8   582.4  5008.3   581.9
    5024   582.4  5031.9   584.6  5047.8  585.79  5095.1  587.09  5137.2  590.05
  5380.5  594.86  5441.2  594.42  5558.6  596.56  5680.7  599.96  5716.1  600.64
#Mann= 8 ,-1 , 0
    4009    .035       0  4321.6     .07       0  4609.7     .05       0
  5007.8     .05       0    5024     .05       0  5380.5     .07       0
  5558.6    .035       0  5680.7     .07       0
Bank Sta=5007.8,5024
XS Rating Curve= 0 ,0
Exp/Cntr=0.3,0.1

Type RM Length L Ch R = 1 ,26753   ,301,301,301
BEGIN DESCRIPTION:
A19800
END DESCRIPTION:
XS GIS Cut Line= 3
       2258135.4     13778302.99      2258788.15     13777844.68
      2259225.64     13776782.21
#Sta/Elev= 30
  4269.7  620.78  4367.9  618.15  4432.8  615.99  4447.7  616.43  4575.8  611.38
    4648  607.55  4676.9  607.43  4684.8   606.4  4697.8  604.39  4727.4  602.85
    4757   599.6  4834.6  594.85  4883.3  590.69    4929  588.42  4965.3   584.7
    5001  584.47  5007.1  581.97  5013.8  581.39  5014.3  580.89  5030.1  581.39
  5036.8  585.31  5082.4  584.85  5196.7  584.61  5380.6  587.85  5522.6  591.93
  5724.6  595.35  5769.9  594.99  5927.1     598  5977.4  599.15  6216.3  604.55
#Mann= 10 ,-1 , 0
  4269.7    .035       0  4367.9     .07       0  4684.8    .035       0
  4883.3     .07       0  5013.8     .05       0  5030.1     .07       0
  5082.4     .05       0  5724.6     .07       0  5927.1    .035       0
  5977.4     .07       0
Bank Sta=5013.8,5030.1
XS Rating Curve= 0 ,0
Exp/Cntr=0.3,0.1

Type RM Length L Ch R = 1 ,26452   ,480,480,480
BEGIN DESCRIPTION:
LONG CREEK 43.0
END DESCRIPTION:
XS GIS Cut Line= 3
        2259025.     13778424.97        2258975.       13778025.
        2259275.     13776825.01
#Sta/Elev= 30
  4591.6  601.79  4795.6  596.56  4833.4   593.7  4944.3  589.21  4956.9  588.57
  4974.5  582.98  4984.6   581.4  5009.4  580.97  5009.9  580.47  5026.4  580.97
  5035.9  584.53  5046.2  585.61  5066.8  584.42  5159.1  584.75    5224  583.92
  5347.7  585.96  5458.5  590.03  5489.4  593.29  5499.8  595.35  5548.7  591.15
  5561.6  592.67    5590   591.1  5609.5  593.05  5631.2   593.9  5736.4   594.5
  5752.6   594.7  5996.9  599.06    6077  601.51    6126  601.76  6231.6  604.31
#Mann= 9 ,-1 , 0
  4591.6     .07       0  5009.4     .05       0  5026.4     .07       0
  5159.1     .05       0  5489.4     .07       0  5609.5    .035       0
  5736.4     .07       0  5752.6    .035       0  5996.9     .07       0
Bank Sta=5009.4,5026.4
XS Rating Curve= 0 ,0
Exp/Cntr=0.3,0.1

Type RM Length L Ch R = 1 ,25972   ,458,458,458
BEGIN DESCRIPTION:
LONG CREEK 42.0
END DESCRIPTION:
XS GIS Cut Line= 3
      2259225.02     13778374.96        2259425.       13777925.
        2259325.     13777125.02
#Sta/Elev= 30
  4503.7   599.1  4580.3  596.95  4686.3  590.91  4853.8  586.48  4906.5  582.96
  4958.5  581.61    4964  582.61  4978.7  578.81  4979.2  578.31  4995.7  578.81
  5006.2  582.79  5072.5  582.94  5167.4  581.92  5179.1   584.7  5187.6  586.53
  5195.1  583.26  5200.2  583.89  5207.7  581.18  5217.8  580.29  5268.2  580.49
  5280.8  583.31  5298.4  583.07  5338.7  586.46  5356.4  588.62  5361.4  590.59
  5379.1  588.92  5392.1  590.84  5457.1   592.7  5788.8  598.68  5802.3  598.91
#Mann= 8 ,-1 , 0
  4503.7     .07       0  4978.7     .05       0  4995.7     .07       0
  5072.5     .05       0  5179.1     .07       0  5392.1     .12       0
  5457.1     .07       0  5788.8    .035       0
Bank Sta=4978.7,4995.7
XS Rating Curve= 0 ,0
Exp/Cntr=0.3,0.1

Type RM Length L Ch R = 1 ,25514   ,458,458,458
BEGIN DESCRIPTION:
LONG CREEK 41.0
END DESCRIPTION:
XS GIS Cut Line= 3
      2259275.02     13778424.97        2259725.       13777825.
        2259725.     13777124.96
#Sta/Elev= 30
  4250.5  600.23  4350.5  596.68  4407.8  592.49  4472.3  590.71  4500.5  591.35
  4522.3  589.84  4593.2   588.7  4628.6  587.32  4636.9  587.85  4672.3   587.2
  4807.8  582.24  4973.9  582.21  4978.6  581.95  4988.8  578.27  4989.3  577.77
  5005.9  578.27  5030.5  581.63  5047.6  582.28  5150.5  580.95  5180.5   584.4
  5200.5  585.81  5260.5     587    5364   591.1  5420.5  592.71  5450.5  594.44
  5560.9  595.98  5595.2  596.81  5660.5  598.39  5690.5  599.91  5700.5  599.49
#Mann= 8 ,-1 , 0
  4250.5     .07       0  4973.9     .12       0  4988.8     .05       0
  5005.9     .12       0  5047.6     .07       0    5364    .035       0
  5560.9     .07       0  5595.2    .035       0
Bank Sta=4988.8,5005.9
XS Rating Curve= 0 ,0
Exp/Cntr=0.3,0.1

Type RM Length L Ch R = 1 ,25056   ,433,433,433
BEGIN DESCRIPTION:
LONG CREEK 40.0
END DESCRIPTION:
XS GIS Cut Line= 3
        2259675.       13778525.        2260025.       13778025.
      2259724.99     13776824.96
#Sta/Elev= 30
  4381.6  598.42  4557.1  592.62  4856.3   584.3  4862.5  584.98  4877.3  583.95
  4948.8  583.54  4963.6  582.14  4969.7  582.96  5002.2  580.11  5006.6  577.71
  5007.1  577.21  5023.7  577.71  5033.2  580.12  5262.5  581.83  5352.7  584.09
  5386.2  583.82  5465.7  586.48  5610.4  591.76  5661.9  592.25  5723.8  595.49
  5734.1  594.77  5857.8  597.41  5875.8  596.79    5881   597.8    5899  597.01
  5917.1  598.24  5929.9  597.74  5958.3  600.05    5991   600.4  6228.9   607.2
#Mann= 6 ,-1 , 0
  4381.6     .05       0  4557.1     .07       0  5006.6     .05       0
  5023.7     .07       0  5465.7    .035       0    5991     .07       0
Bank Sta=5006.6,5023.7
XS Rating Curve= 0 ,0
Exp/Cntr=0.3,0.1

Type RM Length L Ch R = 1 ,24623   ,447,447,447
BEGIN DESCRIPTION:
LONG CREEK 39.0
END DESCRIPTION:
XS GIS Cut Line= 3
      2261424.98     13779024.98        2260325.       13777825.
        2259825.     13776824.99
#Sta/Elev= 30
  3371.4   598.3  3512.9   597.4    3697  597.91  4043.8  595.99  4298.5  592.65
  4390.3  592.37    4607  587.77  4767.9  585.42  4871.9   583.8  4907.1  582.09
  4928.7  582.29    4957   580.5  4963.8  579.31  4971.2  579.42  4976.7  578.26
  4977.2  577.76  4994.1  578.26  4995.9  579.21  5013.2  580.06    5044  580.45
    5058  579.48  5155.8  579.15  5281.6  582.76  5298.3  581.56  5303.9  582.87
  5312.3  581.66  5424.1  586.16  5562.4  590.05  5700.8  595.51  6117.3  607.53
#Mann= 6 ,-1 , 0
  3371.4    .035       0    4607     .07       0  4767.9    .035       0
  4976.7    .035       0  4994.1    .035       0  5562.4     .07       0
Bank Sta=4976.7,4994.1
XS Rating Curve= 0 ,0
Exp/Cntr=0.3,0.1

Type RM Length L Ch R = 1 ,24176   ,413,413,413
BEGIN DESCRIPTION:
LONG CREEK 38.0
END DESCRIPTION:
XS GIS Cut Line= 3
        2260975.       13778425.        2260375.       13777425.
      2260275.01     13777125.02
#Sta/Elev= 30
  3833.4  595.98  3841.2  595.42    3847  596.04  3891.7  594.71    3950  594.46
  4043.3  592.75  4080.2  592.92    4090  592.18  4265.5  588.31  4393.2  584.66
  4482.6  583.27  4721.6     582    4780  578.32  4789.7   578.2  4824.7  579.95
  4927.7  578.47  4991.8  579.15  5002.2   578.9  5010.1  576.16    5012  574.84
  5012.5  574.34  5028.9  574.34  5029.4  574.84  5031.2   577.7  5041.8  578.31
  5052.3  580.62  5073.4   582.9  5083.9  585.69  5126.1  588.77  5315.8  595.66
#Mann= 4 ,-1 , 0
  3833.4    .035       0  4265.5     .07       0    5012     .05       0
  5029.4     .07       0
Bank Sta=5012,5029.4
XS Rating Curve= 0 ,0
Exp/Cntr=0.3,0.1

Type RM Length L Ch R = 1 ,23763   ,496,496,496
BEGIN DESCRIPTION:
LONG CREEK 37.0
END DESCRIPTION:
XS GIS Cut Line= 3
      2261125.01     13778325.03        2260725.       13777325.
      2260525.01     13777025.02
#Sta/Elev= 30
  3922.9  595.67  3967.4  595.43  4014.2  593.94  4067.8  592.48  4153.1   590.6
  4338.9  584.19  4408.2     583  4500.5   580.9  4730.7  580.49    4798  579.35
  4847.8  577.33  4913.8  578.85  4946.1  578.86  4967.7  577.81  4976.5  575.15
    4977  574.65  4993.9  575.15    5003  575.26  5007.5  577.92  5028.5   578.5
  5043.5  581.85  5049.5  581.65  5058.6  583.79  5064.6  582.96  5085.6  586.94
  5094.6  586.94  5100.6  586.01  5121.7  588.55  5223.8  593.25  5360.5  595.99
#Mann= 6 ,-1 , 0
  3922.9    .035       0  4014.2     .07       0  4067.8    .035       0
  4408.2     .07       0  4976.5     .05       0  4993.9     .07       0
Bank Sta=4976.5,4993.9
XS Rating Curve= 0 ,0
Exp/Cntr=0.3,0.1

Type RM Length L Ch R = 1 ,23267   ,918,918,918
BEGIN DESCRIPTION:
A19799
END DESCRIPTION:
XS GIS Cut Line= 3
      2261281.21     13778316.93      2261177.04     13777303.01
      2260650.47      13776499.3
#Sta/Elev= 30
  4102.2  596.03  4186.5  594.08  4366.9  586.99  4453.8  583.49  4503.3  580.65
  4526.3  581.93  4536.4  579.61  4556.5  578.71  4677.1  578.98  4696.7  582.21
  4717.3  583.31  4747.5  577.32  4988.8  577.65  4994.2  575.44  4999.3  577.03
  5010.2  574.77  5010.7  574.27  5027.7  574.77    5039  579.92  5049.1  582.38
  5093.4   585.2  5117.9  583.44  5150.8  584.97  5186.9  583.54    5332  586.49
  5340.2  586.51  5458.5  588.57  5865.2  596.98  6079.5  603.95  6082.3  604.13
#Mann= 10 ,-1 , 0
  4102.2    .035       0  4186.5     .07       0  4366.9    .035       0
  4453.8     .07       0  5010.2     .05       0  5027.7     .07       0
    5332    .035       0  5340.2     .07       0  5458.5    .035       0
  6079.5     .07       0
Bank Sta=5010.2,5027.7
XS Rating Curve= 0 ,0
Exp/Cntr=0.3,0.1

Type RM Length L Ch R = 1 ,22349   ,408,408,408
BEGIN DESCRIPTION:
LONG CREEK 36.0
END DESCRIPTION:
XS GIS Cut Line= 3
        2261675.     13778175.04        2261675.       13777925.
        2260625.     13776125.01
#Sta/Elev= 30
    4750  594.37    4790  592.47    4820  588.35    4860  579.97    4880  577.59
  5002.9  576.49  5007.9  575.28  5013.7  576.29  5014.4  574.53  5014.9  574.03
    5032  574.53  5035.2  575.86  5045.1  576.79  5131.1  577.06  5248.5  579.77
  5510.7  582.74  5590.9  582.53  5665.3  584.43    5767  581.46  5921.7  585.09
  5943.2  584.44  5980.4  586.08  6082.1  585.35  6149.9  586.64  6183.8  586.52
  6312.6  590.37  6385.5  592.94    6632  599.36  6771.1  604.39  7083.9  615.21
#Mann= 7 ,-1 , 0
    4750     .07       0  5014.4     .05       0    5032     .07       0
  6149.9    .035       0  6312.6     .07       0  6385.5    .035       0
  6771.1     .07       0
Bank Sta=5014.4,5032
XS Rating Curve= 0 ,0
Exp/Cntr=0.3,0.1

Type RM Length L Ch R = 1 ,21941   ,626,626,626
BEGIN DESCRIPTION:
LONG CREEK 35.0
END DESCRIPTION:
XS GIS Cut Line= 3
        2262025.     13778225.02        2261975.       13777675.
      2261175.01     13776475.01
#Sta/Elev= 30
    4461  594.01  4467.2  593.86  4566.3   592.5  4712.1  589.39  4732.1   587.4
  4802.4  576.38  4822.5  575.19  4973.1  576.43  4993.2  575.88  5001.9  574.58
  5002.4  574.08  5019.6  574.58  5020.8     576  5056.9  576.54    5165  576.63
  5207.1  577.29  5216.1   578.2  5229.6  577.27  5417.4  582.63  5423.4  582.06
  5525.6  582.82  5567.6  583.81  5576.7  582.97  5597.7  583.87  5705.9  583.02
  5861.4  584.75  6044.5  588.43  6106.4  589.66    6325  594.39  6455.5  597.33
#Mann= 9 ,-1 , 0
    4461     .07       0  4467.2    .035       0  4566.3     .07       0
  5001.9     .05       0  5019.6     .07       0  5861.4    .035       0
  6044.5     .07       0  6106.4    .035       0    6325     .07       0
Bank Sta=5001.9,5019.6
XS Rating Curve= 0 ,0
Exp/Cntr=0.3,0.1

Type RM Length L Ch R = 1 ,21315   ,679,679,679
BEGIN DESCRIPTION:
A19798
END DESCRIPTION:
XS GIS Cut Line= 4
      2262121.47      13778233.6      2262413.15     13777622.45
      2262024.26     13776747.45       2261365.3     13776019.13
#Sta/Elev= 30
  3917.5  593.14  3930.4  592.95    4038  591.32  4115.4  589.21  4412.3  585.33
  4635.7   582.9  4746.6  580.08  4985.9  574.45  4993.9  574.15  4998.9  572.81
  4999.4  572.31  5016.6  572.81  5022.6  574.61  5045.8  575.17  5121.1  573.91
  5160.9  579.75  5196.3   580.3  5294.8  580.74  5312.6  579.87  5318.1  580.56
  5423.6  579.37  5439.8  578.87  5445.5  577.76  5486.3  577.58  5550.8   579.8
  5617.2  580.18  5822.7  587.24  5949.7  593.29  6204.5  598.02  6534.4  606.29
#Mann= 7 ,-1 , 0
  3917.5     .07       0  3930.4    .035       0    4038     .07       0
  4412.3    .035       0  4746.6     .07       0  4998.9     .05       0
  5016.6     .07       0
Bank Sta=4998.9,5016.6
XS Rating Curve= 0 ,0
Exp/Cntr=0.3,0.1

Type RM Length L Ch R = 1 ,20636   ,510,510,510
BEGIN DESCRIPTION:
A19797
END DESCRIPTION:
XS GIS Cut Line= 4
      2262204.84     13778219.64      2262677.04     13777497.45
      2262677.04     13776636.34        2262184.      13775782.2
#Sta/Elev= 30
  3564.6  591.78  3581.8  591.33  3897.3  585.72    4190  582.34  4483.3  581.68
  4749.9  574.33  4779.9   574.8  4819.9  579.06  4854.1  575.63  4959.9  573.87
    4991  571.59  4991.5  571.09  5008.9  571.59  5009.9   573.1  5019.9  575.51
  5209.9  577.44  5229.9  575.94  5239.9  577.23  5336.3  578.89  5532.3  580.86
  5583.6  581.65  5590.3  582.74  5599.4  581.79  5723.1  582.29  5883.8   588.6
  5966.5  593.57  6038.8  597.74  6153.8  602.15  6181.9  603.18  6274.8  606.68
#Mann= 13 ,-1 , 0
  3564.6    .035       0  3581.8     .07       0  3897.3    .035       0
    4190     .07       0  4483.3    .035       0  4854.1     .07       0
    4991     .05       0  5008.9     .07       0  5532.3     .05       0
  5723.1     .07       0  5966.5    .035       0  6153.8     .07       0
  6181.9    .035       0
Bank Sta=4991,5008.9
XS Rating Curve= 0 ,0
Exp/Cntr=0.3,0.1

Type RM Length L Ch R = 1 ,20126   ,939,939,939
BEGIN DESCRIPTION:
LONG CREEK 34.0
END DESCRIPTION:
XS GIS Cut Line= 3
      2262276.69     13778211.44      2263157.77     13777039.56
       2263474.6     13776340.79
#Sta/Elev= 30
    3641  590.64  3707.8  589.36  3909.5  585.51  4037.8  583.74  4282.1  580.67
  4290.8  580.59  4426.6  581.01  4579.7  580.48  4775.2  578.36  4950.5  575.42
  4979.6  573.75  4985.2  570.09  4985.7  569.59  5003.2  570.09  5008.8  572.43
    5015  570.53  5023.3  572.74  5068.2  572.53  5203.7  573.38  5285.9  573.71
  5364.7  576.67  5397.6  580.87  5408.6  584.63  5426.2  585.92  5431.7  588.51
  5473.4  591.83  5570.2  593.97  5650.5  599.26  5737.3  598.78  5874.4  606.18
#Mann= 15 ,-1 , 0
    3641    .035       0  3707.8     .07       0  3909.5    .035       0
  4037.8     .07       0  4282.1    .035       0  4290.8     .07       0
  4426.6    .035       0  4579.7    .045       0  4775.2     .07       0
  4985.2     .05       0  5003.2     .07       0  5068.2     .12       0
  5203.7     .07       0  5285.9     .12       0  5473.4     .07       0
Bank Sta=4985.2,5003.2
XS Rating Curve= 0 ,0
Exp/Cntr=0.3,0.1

Type RM Length L Ch R = 1 ,19187   ,514,514,514
BEGIN DESCRIPTION:
LONG CREEK 33.0
END DESCRIPTION:
XS GIS Cut Line= 3
      2262341.79     13778267.86        2263675.       13777075.
      2263874.99       13777025.
#Sta/Elev= 30
  3215.2  590.14  3313.2  588.29  3390.7   586.3  3603.6  582.25  3625.9  581.73
  3948.1  577.79  4122.2   576.9  4458.7  575.23  4493.7  573.74  4701.3  571.98
    4763   571.3  4834.1  572.55  4884.1  571.75  4961.9  571.61    4967  568.75
  4967.5  568.25  4985.2  568.75  4990.3   573.4  4997.1  574.98  5000.8  579.09
  5006.7  579.09    5016  584.58  5022.2  588.14  5027.3  588.73  5045.4  597.36
  5055.7   601.2  5063.4  602.68  5068.6  602.24  5096.9  606.41  5210.3   612.6
#Mann= 13 ,-1 , 0
  3215.2    .035       0  3313.2     .07       0  3390.7    .045       0
  3603.6     .07       0  3625.9    .045       0  3948.1     .07       0
  4122.2    .045       0  4493.7     .07       0  4701.3     .12       0
  4884.1     .07       0    4967     .05       0  4985.2     .07       0
    5016     .12       0
Bank Sta=4967,4985.2
XS Rating Curve= 0 ,0
Exp/Cntr=0.3,0.1

Type RM Length L Ch R = 1 ,18673   ,372,372,372
BEGIN DESCRIPTION:
LONG CREEK 32.0
END DESCRIPTION:
XS GIS Cut Line= 3
      2262292.55     13778353.12      2263492.53     13777553.13
      2263775.03     13777424.99
#Sta/Elev= 30
  3521.4  592.53  3636.9  589.67  3672.9  589.84  3739.3  587.46  4126.6  579.35
  4365.6  576.79  4415.1     575  4462.4  575.69  4490.7  575.61  4676.5  575.12
  4856.6  572.87  4962.1  570.41  4977.3  571.11  4985.4  565.56  4985.9  565.06
  5003.7  565.56  5010.2   570.4  5023.1  569.66  5032.2  570.51  5046.2  569.81
  5054.2   570.9  5069.3  570.53  5109.1  573.53  5149.7  578.41  5207.8  584.92
  5218.9  584.04  5236.4  588.21  5241.9  587.21  5259.5  591.23  5273.8  592.39
#Mann= 8 ,-1 , 0
  3521.4    .035       0  3739.3    .045       0  4462.4     .07       0
  4490.7    .045       0  4856.6     .07       0  4985.4     .05       0
  5003.7     .07       0  5149.7     .12       0
Bank Sta=4985.4,5003.7
XS Rating Curve= 0 ,0
Exp/Cntr=0.3,0.1

Type RM Length L Ch R = 1 ,18301   ,469,469,469
BEGIN DESCRIPTION:
LONG CREEK 31.0
END DESCRIPTION:
XS GIS Cut Line= 3
      2262824.97     13778575.03        2263525.       13777875.
        2263875.       13777475.
#Sta/Elev= 30
  4005.5  589.94  4118.7  586.56  4191.2  585.49  4373.2  579.64  4571.2  575.02
  4677.3  573.71  4811.6  573.74  4854.1  574.65  4924.8  574.12  4938.9  573.14
  4981.3  573.57    4992  571.38  4998.8  571.38  5007.7  566.53  5008.2  566.03
    5026  566.53  5031.1  569.48  5045.3  570.45  5073.8  570.05  5080.4  570.94
  5137.4  571.67    5144  572.49  5172.5  571.37  5208.1  571.53  5272.2  573.48
    5293  576.36  5336.4  580.51  5370.9  584.63  5434.5  590.12    5527   595.8
#Mann= 5 ,-1 , 0
  4005.5    .035       0  4191.2     .07       0  5007.7     .05       0
    5026     .07       0  5336.4     .12       0
Bank Sta=5007.7,5026
XS Rating Curve= 0 ,0
Exp/Cntr=0.3,0.1

Type RM Length L Ch R = 1 ,17832   ,482,482,482
BEGIN DESCRIPTION:
LONG CREEK 30.0
END DESCRIPTION:
XS GIS Cut Line= 3
        2262675.       13778825.        2263875.       13778125.
      2264075.02     13777724.96
#Sta/Elev= 30
  3615.1  596.06  3761.9  592.98  3817.1  590.83    3940  587.63  3965.2  587.09
    4024  585.54    4067  585.74  4119.9  583.04  4382.1  575.39  4413.5  575.73
  4462.3  574.23  4659.9  572.02  4675.6  573.39  4745.3  574.91  4793.1  576.86
  4798.9  576.07  4814.6  577.26  4851.8  577.14  4916.3  570.61    4975  569.34
  4987.3  566.39  4987.8  565.89  5005.6  566.39  5007.1  568.47  5012.7  569.04
  5102.2  571.44  5175.6  575.13  5236.3  576.95  5364.3  585.59  5451.6  591.65
#Mann= 9 ,-1 , 0
  3615.1    .035       0  3817.1     .07       0    3940    .035       0
  3965.2     .07       0  4745.3     .12       0  4987.3     .05       0
  5005.6     .12       0  5175.6     .07       0  5364.3    .035       0
Bank Sta=4987.3,5005.6
XS Rating Curve= 0 ,0
Exp/Cntr=0.3,0.1

Type RM Length L Ch R = 1 ,17350   ,450,450,450
BEGIN DESCRIPTION:
A19796
END DESCRIPTION:
XS GIS Cut Line= 3
      2264234.16     13779617.65      2264103.95     13778610.74
      2264294.92     13777582.11
#Sta/Elev= 30
  3891.3  587.27  4035.1   584.5    4136  581.27  4209.5  581.01  4307.4   580.3
  4337.6   577.8  4367.9  576.72  4434.8  576.66  4640.1  575.55  4710.7  574.12
  4791.4   571.1  4858.2  570.57  4912.4  568.46  4973.5  569.21  5004.3  565.75
  5004.8  565.25    5024  565.75  5024.3  567.68  5049.5  569.44  5176.9     569
  5295.4  570.56  5339.6  572.41  5400.6  572.36  5492.4  574.79  5644.7  582.95
  5703.7  587.94  5761.6  589.99  5797.3  592.24  5819.5  592.35  5952.8  597.55
#Mann= 6 ,-1 , 0
  3891.3    .035       0  4209.5    .063       0  4434.8    .035       0
  5004.3    .035       0    5024    .035       0  5295.4     .07       0
Bank Sta=5004.3,5024
XS Rating Curve= 0 ,0
Exp/Cntr=0.3,0.1

Type RM Length L Ch R = 1 ,16900   ,391,391,391
BEGIN DESCRIPTION:
LONG CREEK 29.0
END DESCRIPTION:
XS GIS Cut Line= 3
      2264874.99     13779424.98        2264551.     13778719.24
        2264375.     13777425.01
#Sta/Elev= 30
    4128  588.45    4647  574.45  4777.2  572.13  4836.4  573.32  4882.4   571.1
  4912.9  572.35    4929  570.47  4949.2     566  4959.3  565.42  4979.5  566.73
  4980.6  564.35  4981.1  563.85  5000.3  564.35  5009.8  566.95  5028.1  568.37
  5062.8  568.88  5120.8  572.55  5135.3  574.56    5151  574.81  5201.5  574.51
  5221.7  571.59    5252  570.46  5507.5  573.81  5746.5  584.11  5766.7  583.85
  5874.7  588.87  5879.7  588.25    5918   591.5  5998.8  595.22  6210.7   603.2
#Mann= 4 ,-1 , 0
    4128    .035       0  4980.6    .035       0  5000.3    .035       0
  5028.1     .07       0
Bank Sta=4980.6,5000.3
XS Rating Curve= 0 ,0
Exp/Cntr=0.3,0.1

Type RM Length L Ch R = 1 ,16509   ,458,458,458
BEGIN DESCRIPTION:
LONG CREEK 28.0
END DESCRIPTION:
XS GIS Cut Line= 3
        2265125.       13779075.        2264875.       13778725.
      2264575.01     13777525.05
#Sta/Elev= 30
  4564.5  581.86    4599  580.83  4658.6  578.59  4761.6  575.54  4859.4  574.53
  4922.1  572.96  4972.5  570.46  4997.2  567.83  5004.9     566  5015.7  561.29
  5016.2  560.79  5035.4  561.29  5035.8  563.23  5046.8   566.2  5100.3  566.65
  5125.6  568.36  5211.1  567.48    5425  570.36  5471.3  572.36  5548.8   572.6
  5636.3  573.77  5664.6  575.86  5677.5  578.12  5713.6  579.43  5754.8  578.92
    5760  577.73  5767.7  577.75  5870.8  582.84  5932.6  586.96  6231.5  598.25
#Mann= 9 ,-1 , 0
  4564.5     .07       0    4599    .035       0  4658.6     .07       0
  4761.6    .035       0  5015.7    .035       0  5035.4    .035       0
  5046.8     .07       0  5125.6    .035       0  5548.8     .07       0
Bank Sta=5015.7,5035.4
XS Rating Curve= 0 ,0
Exp/Cntr=0.3,0.1

Type RM Length L Ch R = 1 ,16051   ,474,474,474
BEGIN DESCRIPTION:
LONG CREEK 27.0
END DESCRIPTION:
XS GIS Cut Line= 3
      2265425.01     13778925.01        2265275.       13778575.
        2264775.       13777375.
#Sta/Elev= 30
  4614.9  581.79  4658.4  580.01  4676.6  578.29  4793.4  575.58    4905  572.63
  4941.3  567.34  4952.2   567.8  4973.9     565  4976.7  559.56  4977.2  559.06
  4996.5  559.56  5004.9  564.25  5017.4  566.06  5034.2   567.2  5049.9  566.25
  5085.8  566.61  5140.3  567.36  5189.2  566.13  5211.8  565.25  5301.1  567.34
    5474   570.3    5624   572.6  5775.7  578.09  5891.1  584.34  5896.5  583.35
  5965.1  585.37  6003.2  590.29  6074.2  591.12  6103.4  594.11  6295.7  600.98
#Mann= 9 ,-1 , 0
  4614.9     .07       0  4793.4     .12       0  4976.7     .05       0
  4996.5     .12       0  5085.8     .07       0  5189.2    .035       0
  5301.1     .07       0    5474    .035       0  5965.1     .07       0
Bank Sta=4976.7,4996.5
XS Rating Curve= 0 ,0
Exp/Cntr=0.3,0.1

Type RM Length L Ch R = 1 ,15577   ,452,452,452
BEGIN DESCRIPTION:
LONG CREEK 26.0
END DESCRIPTION:
XS GIS Cut Line= 3
      2265725.02     13778775.04        2265375.       13778175.
      2265175.01     13777575.02
#Sta/Elev= 30
  4297.5  580.07  4342.6  579.07  4348.4  578.17  4385.6   576.7  4436.5  576.24
  4450.1  575.25  4487.3  574.69    4503  573.24  4540.2  573.41  4552.2  572.35
  4700.7  568.29  4737.5  568.33  4749.5  567.54  4853.2  565.78  4866.9  566.78
  4882.6  565.61  4903.6  565.77  4994.8   564.6  5002.7  564.06  5013.2     562
  5013.9  559.76  5014.4  559.26  5033.7  559.76  5034.3  561.16  5097.6  563.63
  5129.2  567.13  5160.8  567.53  5414.9  578.18  5508.7  583.45  5624.6  588.82
#Mann= 5 ,-1 , 0
  4297.5     .12       0  4903.6     .07       0  5013.9     .05       0
  5033.7     .07       0  5414.9    .035       0
Bank Sta=5013.9,5033.7
XS Rating Curve= 0 ,0
Exp/Cntr=0.3,0.1

Type RM Length L Ch R = 1 ,15125   ,469,469,469
BEGIN DESCRIPTION:
LONG CREEK 25.0
END DESCRIPTION:
XS GIS Cut Line= 3
        2265875.     13778724.98        2265725.       13778125.
        2265625.     13777525.02
#Sta/Elev= 30
  4376.4  580.43  4386.7  580.56    4482  576.85  4551.6  576.61  4564.5  575.96
  4572.2  574.45    4683  571.94    4799  566.55  4829.9  567.33  4840.2  566.99
    4848  565.77  4853.1   566.2  4894.3  564.74  4921.1  566.24  4935.6  567.05
  4971.7  563.24  4997.4  561.86    5005  559.53  5005.2  558.53  5005.7  558.03
  5024.6  558.03  5025.1  558.53  5035.4  561.44  5045.5  565.95  5075.1  565.41
  5206.9   568.5  5359.8  572.36  5435.6  577.39  5509.3  583.18  5603.1  589.43
#Mann= 7 ,-1 , 0
  4376.4     .07       0  4921.1     .12       0  5005.2     .05       0
  5025.1     .12       0  5075.1     .07       0  5206.9    .035       0
  5435.6     .07       0
Bank Sta=5005.2,5025.1
XS Rating Curve= 0 ,0
Exp/Cntr=0.3,0.1

Type RM Length L Ch R = 1 ,14656   ,427,427,427
BEGIN DESCRIPTION:
LONG CREEK 24.0
END DESCRIPTION:
XS GIS Cut Line= 3
        2266075.     13778674.96        2266125.       13778125.
        2266175.     13777525.01
#Sta/Elev= 30
  4447.8  578.13  4688.8  576.03  4833.1  572.57  4889.6  570.53  4919.7  568.36
  4929.7  567.25  4939.8   565.1  4949.8  565.82  4953.1  565.43    4990  561.92
  4997.5  559.59    5000  559.59  5000.1   557.8  5000.6   557.3  5019.5   557.3
    5020   557.8  5030.1  558.68  5040.2  562.62  5050.2  564.94  5062.7  564.37
  5090.3  565.34  5110.4  563.46  5128.7  563.09  5183.2  564.13  5303.6  568.66
  5375.2  572.14    5424  574.67  5473.7   578.4  5550.4  583.29  5602.1  587.27
#Mann= 9 ,-1 , 0
  4447.8    .035       0  4833.1     .07       0  4953.1     .12       0
  5000.1     .05       0    5020     .12       0  5128.7     .07       0
  5375.2    .035       0  5473.7     .07       0  5550.4    .035       0
Bank Sta=5000.1,5020
XS Rating Curve= 0 ,0
Exp/Cntr=0.3,0.1

Type RM Length L Ch R = 1 ,14229   ,443,443,443
BEGIN DESCRIPTION:
LONG CREEK 23.0
END DESCRIPTION:
XS GIS Cut Line= 3
      2266174.98     13778725.04        2266475.       13777925.
        2266475.     13777525.05
#Sta/Elev= 30
  4140.9  577.65  4387.5  575.68  4685.2  571.83  4754.2  570.42  4792.4  568.39
  4839.6  567.21  4864.5  564.46  4888.5  563.94  4961.1  564.39    4974  563.62
  4980.2  562.48  4985.6  562.94  4992.7  559.48  4997.8  559.48  5005.3  558.29
  5005.4  557.76  5005.9  557.26  5024.8  557.26  5025.3  557.76  5035.3  561.02
  5045.3  562.92  5055.3  563.87  5085.3   564.2  5159.7   567.6  5225.3  575.21
  5245.3  576.89  5255.3  578.86  5295.3  584.21  5355.3  587.53  5395.3   592.3
#Mann= 6 ,-1 , 0
  4140.9    .035       0  4685.2     .07       0  4961.1     .12       0
  5005.4     .05       0  5025.3     .12       0  5159.7    .035       0
Bank Sta=5005.4,5025.3
XS Rating Curve= 0 ,0
Exp/Cntr=0.3,0.1

Type RM Length L Ch R = 1 ,13786   ,464,464,464
BEGIN DESCRIPTION:
LONG CREEK 22.0
END DESCRIPTION:
XS GIS Cut Line= 3
        2266375.       13778575.        2266875.       13777875.
        2266825.     13777475.04
#Sta/Elev= 30
  4139.7  575.71  4483.8  572.18    4622  569.36  4799.6  565.42  4814.4  565.64
  4820.5  566.56  4827.9  565.09  4841.3  564.79  4864.7  564.65    4877   563.5
  4906.5  562.36  4963.1  562.38  4977.8   561.1  4986.4  558.76  4999.9  556.91
  5000.1  556.24  5000.6  555.74  5019.5  555.74    5020  556.24  5020.5  556.77
  5037.7  562.46  5115.9  566.67    5204  574.27    5272   583.6  5279.6  585.26
  5332.5  591.45  5342.6  591.53  5360.2  594.61  5365.2  594.52    5403  598.93
#Mann= 7 ,-1 , 0
  4139.7    .035       0    4622     .07       0  4841.3    .035       0
  5000.1    .035       0    5020    .035       0  5020.5     .07       0
  5115.9    .035       0
Bank Sta=5000.1,5020
XS Rating Curve= 0 ,0
Exp/Cntr=0.3,0.1

Type RM Length L Ch R = 1 ,13322   ,525,525,525
BEGIN DESCRIPTION:
LONG CREEK 21.0
END DESCRIPTION:
XS GIS Cut Line= 3
      2266625.03     13778724.97        2267325.       13777925.
      2267374.99     13777725.03
#Sta/Elev= 30
  3941.4  575.26  4203.8  573.53  4416.4  570.34  4529.3  569.73  4551.2  568.21
  4565.4  568.83  4586.3  571.42  4614.8  567.48  4643.2     566  4784.7   565.5
  4855.8  561.49    4891  561.24  4919.4   562.6  4940.3  561.78  4947.9   558.9
  4962.1  555.86    4973  555.35  4973.5  554.85    4993  555.35  4997.3  557.27
  5001.1  561.48  5027.6  562.62  5086.8  572.92  5117.8  584.48  5138.4  589.83
  5146.1     593  5151.3   593.9    5159  597.07  5179.6  602.88  5210.5  607.47
#Mann= 3 ,-1 , 0
  3941.4    .035       0    4973    .035       0    4993    .035       0
Bank Sta=4973,4993
XS Rating Curve= 0 ,0
Exp/Cntr=0.3,0.1

Type RM Length L Ch R = 1 ,12797   ,597,597,597
BEGIN DESCRIPTION:
LONG CREEK 20.0
END DESCRIPTION:
XS GIS Cut Line= 3
      2267125.02     13779674.96        2267675.       13778275.
        2267725.     13777824.99
#Sta/Elev= 30
  3483.9  582.55  3655.8  580.55  3829.4  575.13    4076  570.04  4317.3  569.08
  4364.9  567.18  4405.9  568.01  4455.5  568.61  4485.2  567.17  4515.3  571.88
  4539.5  568.63  4569.2   568.7  4618.1  565.34  4672.1  564.35  4715.9  563.34
  4773.1  563.08  4816.1  560.69  4894.5   559.1  4998.1  559.32  5028.3  555.99
  5028.8  555.49  5048.3  555.99  5048.4  557.65  5118.8  562.78  5138.9  565.52
  5189.2  575.77  5269.7  584.77  5314.1  592.47  5400.5  610.45  5440.8  614.14
#Mann= 7 ,-1 , 0
  3483.9     .07       0  4405.9    .035       0  4672.1     .05       0
  4715.9    .035       0  5028.3    .035       0  5048.3    .035       0
  5314.1     .12       0
Bank Sta=5028.3,5048.3
XS Rating Curve= 0 ,0
Exp/Cntr=0.3,0.1

Type RM Length L Ch R = 1 ,12200   ,535,535,535
BEGIN DESCRIPTION:
LONG CREEK 19.0
END DESCRIPTION:
XS GIS Cut Line= 3
      2267524.98     13779775.03        2268075.       13778675.
      2268325.01     13778174.99
#Sta/Elev= 30
  3775.5  580.68  4134.9     568  4201.1  562.86  4231.1  564.72  4401.8  560.85
  4460.3  559.73  4513.4  562.28  4577.4   560.2  4652.4  558.54  4728.7  556.34
  4795.7   564.3  4862.8  564.21    4902  559.31    4969  560.23    4983  557.81
  4985.6  555.16    4987  553.74  4987.5  553.24    5007  553.74  5036.1  561.84
  5092.9  567.22  5165.7  570.62  5265.3   586.1  5393.9  587.97  5438.6  593.43
  5463.2  599.24  5488.9  605.07  5519.7  616.55  5526.6  616.34  5564.4  615.94
#Mann= 13 ,-1 , 0
  3775.5     .12       0  4134.9     .07       0  4201.1     .12       0
  4401.8    .035       0  4577.4     .05       0  4652.4    .035       0
  4985.6     .05       0    4987    .035       0    5007     .05       0
  5092.9     .05       0  5165.7    .035       0  5463.2     .05       0
  5526.6    .035       0
Bank Sta=4987,5007
XS Rating Curve= 0 ,0
Exp/Cntr=0.3,0.1

Type RM Length L Ch R = 1 ,11665   ,547,547,547
BEGIN DESCRIPTION:
LONG CREEK 18.0
END DESCRIPTION:
XS GIS Cut Line= 3
      2267774.99     13779775.02        2268175.       13779175.
      2268725.03     13778374.96
#Sta/Elev= 30
  4274.9  580.41  4441.7  571.94  4585.9  567.99    4628  562.25    4658  554.69
  4724.3  558.92  4779.7     559  4823.3  562.02  4859.3   557.2  4973.5  556.59
  4982.5  555.24    4983  552.94  4983.5  552.44    5003  552.94  5126.8  559.67
  5218.6  559.69  5239.6  561.19  5248.4  564.96  5290.3  562.04  5341.1  567.97
    5356  565.17  5427.7  566.27  5642.8  581.66  5693.5  586.87  5736.3  594.73
  5798.6  599.28  5866.7  600.97  5902.6  606.46  5930.4  613.86  5966.9  614.63
#Mann= 6 ,-1 , 0
  4274.9     .12       0  4724.3    .035       0    4983    .035       0
    5003    .035       0  5126.8     .05       0  5798.6    .035       0
Bank Sta=4983,5003
XS Rating Curve= 0 ,0
Exp/Cntr=0.3,0.1

Type RM Length L Ch R = 1 ,11118   ,591,591,591
BEGIN DESCRIPTION:
LONG CREEK 17.0
END DESCRIPTION:
XS GIS Cut Line= 3
        2267825.       13779825.        2268425.       13779475.
        2269075.       13779325.
#Sta/Elev= 30
  4305.9  580.26  4502.7  571.58    4752  565.77  4773.5  563.96  4785.2  561.18
    4787  560.69    4795  557.98  4847.9  558.56  4869.5  555.47    4903   557.4
  4968.8   556.8  4987.6  551.03  4988.1  550.53  5007.7  551.03  5016.8  554.39
  5051.8  556.82    5110  558.57  5227.3  555.06  5269.5  554.52  5291.3  554.05
  5318.7  555.86  5328.9  554.85  5349.5  558.67    5370  559.77  5423.9  559.38
  5482.9  559.03    5553  587.17    5592  596.36  5636.8  602.45  5667.6  603.05
#Mann= 12 ,-1 , 0
  4305.9     .12       0  4785.2    .035       0    4787     .12       0
    4903     .07       0  4968.8    .035       0  4987.6    .035       0
  5007.7    .035       0  5016.8     .05       0  5227.3    .035       0
  5269.5     .05       0  5423.9     .12       0    5592     .05       0
Bank Sta=4987.6,5007.7
XS Rating Curve= 0 ,0
Exp/Cntr=0.3,0.1

Type RM Length L Ch R = 1 ,10527   ,528,528,528
BEGIN DESCRIPTION:
LONG CREEK 16.0
END DESCRIPTION:
XS GIS Cut Line= 3
        2268425.       13780125.        2268775.       13779925.
      2269025.01     13779374.97
#Sta/Elev= 30
  4592.3  571.73  4685.5   569.7  4818.9   567.4  4862.6  565.96  4922.7   563.5
  4960.1  557.71  4972.4  552.67  4982.4  544.51  4982.9  544.01  5002.6  544.51
  5009.7  550.62  5017.4  551.71  5050.3  549.13  5070.6  550.32  5227.4  551.67
  5268.9  549.77  5322.6   551.8  5389.8  553.28  5441.4  558.54  5446.9  565.17
  5464.5  565.63  5469.9  572.51  5487.5   576.6    5493  583.69  5510.6  587.78
  5516.1  598.75  5543.3  600.33  5562.2  598.96  5589.6  603.33  5599.6  604.32
#Mann= 11 ,-1 , 0
  4592.3      .1       0  4685.5     .12       0  4818.9      .1       0
  4862.6     .07       0  4982.4     .05       0  5002.6     .07       0
  5070.6    .035       0  5227.4     .05       0  5322.6    .035       0
  5543.3     .12       0  5589.6     .05       0
Bank Sta=4982.4,5002.6
XS Rating Curve= 0 ,0
Exp/Cntr=0.3,0.1

Type RM Length L Ch R = 1 ,9999    ,531,531,531
BEGIN DESCRIPTION:
LONG CREEK 15.0
END DESCRIPTION:
XS GIS Cut Line= 3
      2269325.02     13780675.04        2269125.       13780275.
        2269025.     13779474.99
#Sta/Elev= 30
  4548.2   568.4  4619.1  569.36    4632  569.25  4743.7   565.6  4785.8  564.72
  4826.9  561.14  4860.4  561.18  4875.3  561.63  4936.8  555.49  4987.1  554.12
  4995.2   542.8  4995.7   542.3  5015.8   542.8  5025.7  545.42  5033.3   550.5
  5038.3  548.54  5045.8   551.1  5076.1  553.06  5166.8  552.56  5348.4  557.38
  5453.3  559.88    5522  562.85  5602.6  569.31  5660.6  576.97  5697.1  583.87
  5758.9  595.47  5763.9  594.52  5781.5  596.94  5796.9  601.09  5801.7  601.92
#Mann= 12 ,-1 , 0
  4548.2    .035       0  4619.1      .1       0    4632    .035       0
  4743.7     .05       0  4826.9      .1       0  4860.4    .035       0
  4995.2    .035       0  5015.8    .035       0  5348.4     .05       0
  5453.3    .035       0  5697.1     .05       0  5796.9    .035       0
Bank Sta=4995.2,5015.8
XS Rating Curve= 0 ,0
Exp/Cntr=0.3,0.1

Type RM Length L Ch R = 1 ,9468    ,315,315,315
BEGIN DESCRIPTION:
LONG CREEK 14.0
END DESCRIPTION:
XS GIS Cut Line= 3
        2269675.     13780675.01        2269625.       13780275.
      2269075.03     13779475.04
#Sta/Elev= 30
  4592.7  571.96  4656.8  571.75  4683.4  571.98  4703.6  568.27  4723.7  570.61
  4756.4   569.3  4824.5  567.65  4844.7   562.7  4872.4  559.89    4958  558.97
  4985.7  551.93    4993  541.56  4993.5  541.06  5013.6  541.56  5024.2  543.86
  5032.2  548.34  5068.6  548.22  5125.7     552  5293.8  557.91  5427.5  562.99
  5627.7  563.98  5779.9  569.06  5815.8  572.76  5857.7  580.96  5887.5   583.5
  5913.5  588.69  5923.3  592.04  5938.2  593.39  5944.3  595.63  5966.6  596.21
#Mann= 7 ,-1 , 0
  4592.7    .035       0  4656.8     .05       0  4756.4    .035       0
    4993    .035       0  5013.6    .035       0  5293.8     .05       0
  5913.5    .035       0
Bank Sta=4993,5013.6
XS Rating Curve= 0 ,0
Exp/Cntr=0.3,0.1

Type RM Length L Ch R = 1 ,9153    ,247,247,247
BEGIN DESCRIPTION:
A19795
END DESCRIPTION:
XS GIS Cut Line= 3
      2270054.48     13780620.29      2269789.72     13780056.05
      2269130.02     13779470.13
#Sta/Elev= 30
  4344.1  570.73  4423.5  570.56  4446.3  569.79  4460.4  568.02  4482.5   568.8
  4617.1  567.62    4754  564.99  4822.4  562.05  4845.2  559.91  4850.8  556.96
  4858.1  558.76  4868.1  559.38  4924.7  551.77  4947.6   550.8  4957.5  548.41
  4968.1  540.55  4968.6  540.05  4988.7  540.55  4992.6  545.06  5000.2  551.18
  5006.9   552.5  5063.7   554.7  5092.2  553.34  5098.8  555.87  5113.1  558.63
  5141.5  562.25  5594.7  564.74  5651.6  565.82  5722.7  569.28  5849.7  591.21
#Mann= 3 ,-1 , 0
  4344.1    .035       0  4968.1    .035       0  4988.7    .035       0
Bank Sta=4968.1,4988.7
XS Rating Curve= 0 ,0
Exp/Cntr=0.3,0.1

Type RM Length L Ch R = 1 ,8906    ,551,551,551
BEGIN DESCRIPTION:
LONG CREEK 13.0
END DESCRIPTION:
XS GIS Cut Line= 3
        2270225.       13780025.        2269875.       13779825.
        2269075.       13779375.
#Sta/Elev= 30
  4597.4  568.87  4772.3  566.64  4919.9  557.98  4977.5  552.33  4992.6  549.43
  4997.6  542.59  5003.4  542.59  5003.9  538.63  5004.4  538.13  5024.5  538.63
  5030.2  547.48  5035.9   545.9  5046.1  548.87  5095.2  551.79  5111.1  555.03
  5116.8  553.91  5128.2     557  5130.1  557.86  5132.8  559.07  5138.5  557.91
  5161.1  562.34  5197.8  563.93  5397.3  566.09  5580.9  564.93  5667.6  567.62
  5705.2  570.02  5780.4  582.91  5845.4  596.66    5902  603.17  5918.4  604.85
#Mann= 6 ,-1 , 0
  4597.4    .035       0  5003.9    .035       0  5024.5    .035       0
  5128.2     .05       0  5130.1    .035       0    5902     .05       0
Bank Sta=5003.9,5024.5
XS Rating Curve= 0 ,0
Exp/Cntr=0.3,0.1
