HEC-RAS study West Fork Dry Comal Creek.prj: West Fork Dry Comal Creek

--- West Fork Dry Comal Creek.g01 (geometry) --- (continued)

Type RM Length L Ch R = 1 ,74287   ,451,451,451
BEGIN DESCRIPTION:
West Fork 126.0
END DESCRIPTION:
XS GIS Cut Line= 3
      2183075.01     13825675.01        2182075.       13824475.
      2181875.01     13824225.01
#Sta/Elev= 30
  3432.9 1146.09  3610.6 1134.42  3849.8 1128.49  3991.5 1127.74  4088.9 1127.42
    4244 1127.13  4373.8 1126.58  4469.7 1126.34  4682.4 1121.71  4831.3 1119.84
  4911.4 1118.52  4952.7 1114.88  4959.2  1111.1    4973 1109.27  4973.5 1108.77
  4989.6 1109.27  5002.2 1109.87  5016.6 1113.43  5037.4 1114.42  5045.4 1113.61
  5051.8 1111.03    5059 1110.97  5066.2 1112.38    5095 1112.13  5144.6 1114.54
    5159 1118.05  5215.1 1142.29  5243.9 1152.24  5264.7 1157.61  5315.1  1162.7
#Mann= 11 ,-1 , 0
  3432.9     .12       0  3849.8     .07       0  3991.5     .12       0
  4088.9     .07       0    4244    .035       0  4373.8     .07       0
  4682.4    .035       0  4831.3     .07       0  4911.4     .12       0
    4973     .05       0  4989.6     .12       0
Bank Sta=4973,4989.6
XS Rating Curve= 0 ,0
Exp/Cntr=0.3,0.1

Type RM Length L Ch R = 1 ,73836   ,449,449,449
BEGIN DESCRIPTION:
West Fork 125.0
END DESCRIPTION:
XS GIS Cut Line= 3
      2182574.98     13824974.96        2182175.       13824075.
        2181975.       13824125.
#Sta/Elev= 30
  4021.5 1126.78  4059.1  1127.1  4098.1  1125.6  4135.5  1125.7  4427.4  1120.8
  4620.2 1119.13  4775.2 1117.63    4795 1117.27  4800.5 1115.89  4831.3 1112.74
    4886 1113.33    4940 1111.88  4962.6 1110.45  4974.2 1107.07  4989.2 1104.58
  4989.7 1104.08  5005.8 1104.58  5024.4 1108.88  5029.5 1107.35  5037.3 1110.21
  5065.6 1125.38  5070.8 1123.11  5078.5 1127.55  5099.1 1136.47  5106.8 1141.96
    5112 1140.15  5119.7  1144.9  5148.1 1150.68  5189.5 1154.61  5212.5 1156.34
#Mann= 8 ,-1 , 0
  4021.5    .035       0  4135.5     .07       0  4427.4    .035       0
  4620.2     .07       0  4775.2     .12       0  4989.2     .05       0
  5005.8     .12       0  5189.5     .07       0
Bank Sta=4989.2,5005.8
XS Rating Curve= 0 ,0
Exp/Cntr=0.3,0.1

Type RM Length L Ch R = 1 ,73387   ,454,454,454
BEGIN DESCRIPTION:
West Fork 124.0
END DESCRIPTION:
XS GIS Cut Line= 3
        2182525.     13824725.03        2182525.       13823825.
      2182274.99       13823725.
#Sta/Elev= 30
    4100 1122.74    4110 1122.97    4170 1121.55  4472.6 1118.66  4620.5 1117.39
  4621.2 1117.38    4760 1116.68    4840 1114.34    4910 1111.08  4919.9 1109.98
    4940 1108.65    4960 1106.23    4970 1106.21  4988.8 1102.28  4989.3 1101.78
  5005.7 1101.78  5006.2 1102.28  5014.8    1104  5039.1 1105.36  5044.5 1109.11
  5053.9 1110.81  5063.3 1111.64  5068.7 1113.72  5086.2 1115.42  5117.2 1117.53
  5176.4 1119.24  5200.6 1121.12    5206 1120.47  5254.5 1123.96  5269.3 1124.36
#Mann= 7 ,-1 , 0
    4100     .07       0  4472.6    .035       0  4620.5     .07       0
  4621.2    .035       0  4919.9     .07       0  4988.8     .05       0
  5006.2     .07       0
Bank Sta=4988.8,5006.2
XS Rating Curve= 0 ,0
Exp/Cntr=0.3,0.1

Type RM Length L Ch R = 1 ,72933   ,446,446,446
BEGIN DESCRIPTION:
West Fork 123.0
END DESCRIPTION:
XS GIS Cut Line= 3
        2182975.     13824025.01        2182925.       13823675.
        2182925.     13823474.96
#Sta/Elev= 30
  4641.4 1118.44  4671.7 1118.62  4712.1  1117.7  4732.3 1116.65  4772.7 1115.51
  4782.8 1114.98    4803 1112.95  4823.2  1112.1  4843.4  1112.2  4893.9 1109.67
  4914.1 1109.27  4924.2 1108.13  4954.6 1102.88  4964.7 1101.95  4984.9 1101.59
  4992.4 1099.66    4995 1099.66  4996.2 1098.71  4996.7 1098.21  5013.2 1098.21
  5013.7 1098.71    5035 1103.01    5045 1106.06    5055 1110.59    5075 1116.79
  5084.6 1119.33    5125 1124.59    5155 1126.87    5175 1127.35    5195 1128.64
#Mann= 4 ,-1 , 0
  4641.4     .07       0  4996.2     .05       0  5013.7     .07       0
  5084.6     .12       0
Bank Sta=4996.2,5013.7
XS Rating Curve= 0 ,0
Exp/Cntr=0.3,0.1

Type RM Length L Ch R = 1 ,72487   ,480,480,480
BEGIN DESCRIPTION:
West Fork 122.0
END DESCRIPTION:
XS GIS Cut Line= 3
        2183275.     13823925.01        2183325.       13823525.
        2183325.     13823325.02
#Sta/Elev= 30
  4601.8 1118.11  4652.2 1116.21  4740.7  1113.9  4783.2 1112.41  4805.9 1111.14
  4813.4 1110.12  4839.5 1109.06  4873.9 1107.95  4881.5 1107.18  4886.5 1107.36
  4934.4 1099.91  4944.5 1097.34  4962.1 1096.61  4967.1  1097.1  4974.7 1096.24
    4986 1095.97  4986.5 1095.47  5003.1 1095.47  5003.6 1095.97  5004.9 1096.58
  5007.4 1096.58    5037 1108.95  5054.9 1114.43  5064.9  1116.9  5074.9 1118.38
  5094.9 1122.99  5104.9 1124.72  5124.9 1127.78  5144.9 1129.07  5204.9  1134.9
#Mann= 6 ,-1 , 0
  4601.8     .12       0  4740.7    .035       0  4839.5     .07       0
    4986     .05       0  5003.6     .07       0    5037     .12       0
Bank Sta=4986,5003.6
XS Rating Curve= 0 ,0
Exp/Cntr=0.3,0.1

Type RM Length L Ch R = 1 ,72007   ,486,486,486
BEGIN DESCRIPTION:
West Fork 121.0
END DESCRIPTION:
XS GIS Cut Line= 3
      2183374.98     13824225.03        2183775.       13823425.
        2183575.       13823225.
#Sta/Elev= 30
  4100.9 1120.45  4270.9 1119.02    4472 1116.19  4565.9 1114.66  4580.4 1114.08
  4623.6 1112.13  4688.8 1110.96    4741 1109.81  4763.4 1108.27  4800.3 1103.08
  4824.9 1100.41  4847.2 1103.03  4869.6 1103.05  4897.5 1102.66  4914.3 1100.44
  4919.9 1101.54  4936.7 1100.38  4998.9 1100.65  5014.8 1099.54  5015.3 1099.04
  5032.4 1099.54  5037.8 1101.32  5066.1 1105.39  5094.4 1113.42  5108.5 1116.22
  5193.4 1125.46  5207.5 1126.31  5235.8 1131.97  5249.9 1133.77  5278.2  1135.4
#Mann= 9 ,-1 , 0
  4100.9    .035       0  4270.9     .12       0    4472     .07       0
  4565.9    .035       0  4580.4     .07       0  4688.8    .035       0
  4800.3     .07       0  5014.8     .05       0  5032.4     .12       0
Bank Sta=5014.8,5032.4
XS Rating Curve= 0 ,0
Exp/Cntr=0.3,0.1

Type RM Length L Ch R = 1 ,71521   ,450,450,450
BEGIN DESCRIPTION:
West Fork 120.0
END DESCRIPTION:
XS GIS Cut Line= 3
      2183855.06     13823889.23        2184225.       13823325.
      2183889.58     13822725.33
#Sta/Elev= 30
  4325.3 1114.17    4460 1111.28  4501.1  1111.8  4531.3 1110.16  4660.9 1107.73
  4748.3 1103.28  4805.6 1101.68  4892.4 1102.28  4956.3 1101.42  4977.3 1102.24
  4988.2    1101  4988.7  1100.5  5005.8    1101  5089.1 1103.46  5170.1 1103.67
  5197.6 1108.42  5235.8 1111.12  5252.3 1112.09  5272.9    1113  5278.6  1114.3
  5316.3 1115.22    5338  1117.3  5381.4  1118.3  5397.4 1117.18  5403.1 1118.66
  5412.5 1118.55  5424.8  1120.8  5484.2  1125.2  5581.2 1128.84  5687.1 1136.89
#Mann= 6 ,-1 , 0
  4325.3     .12       0    4460     .07       0  4988.2     .05       0
  5005.8     .07       0  5235.8    .035       0  5252.3     .07       0
Bank Sta=4988.2,5005.8
XS Rating Curve= 0 ,0
Exp/Cntr=0.3,0.1

Type RM Length L Ch R = 1 ,71071   ,433,433,433
BEGIN DESCRIPTION:
West Fork 119.0
END DESCRIPTION:
XS GIS Cut Line= 3
      2185224.99     13823724.99        2184625.       13823175.
      2184125.02     13822625.02
#Sta/Elev= 30
  4191.2 1139.67  4261.8 1134.51    4375 1128.79  4417.8 1123.42    4432  1116.5
  4467.1 1107.24  4481.3 1097.13  4486.6 1092.27  4487.1 1091.77  4504.3 1092.27
  4523.9 1098.94  4545.8 1100.54  4609.1  1102.2  4664.8 1103.21  4797.3 1104.02
    4892 1102.97  4941.3 1096.05  4991.3 1094.64  5033.2 1098.66    5069 1096.65
  5089.9 1097.03  5118.3 1100.16  5139.9 1103.99  5160.9 1105.55  5472.1 1112.07
    5483 1113.19  5507.5 1115.45  5677.8  1124.1  5706.2 1127.77  5748.4 1129.88
#Mann= 10 ,-1 , 0
  4191.2     .07       0    4375     .12       0  4486.6     .05       0
  4504.3     .12       0  4545.8    .035       0  4609.1     .07       0
  4664.8    .035       0  4797.3     .07       0  5472.1    .035       0
    5483     .07       0
Bank Sta=4486.6,4504.3
XS Rating Curve= 0 ,0
Exp/Cntr=0.3,0.1

Type RM Length L Ch R = 1 ,70638   ,422,422,422
BEGIN DESCRIPTION:
West Fork 118.0
END DESCRIPTION:
XS GIS Cut Line= 3
      2185625.04     13823425.02        2185025.       13823075.
        2184425.       13822575.
#Sta/Elev= 30
  4310.6 1153.68  4441.7 1139.96  4463.2 1133.15  4484.7 1121.48  4500.4 1116.76
  4516.1 1114.47  4559.1 1115.52  4574.9 1111.74  4580.6 1112.77  4596.4 1108.62
  4602.1 1109.28  4617.9 1106.55  4639.4 1106.28  4778.3 1095.82  4843.2 1094.22
  4874.2 1098.99  4992.7 1092.72  4993.2 1092.22    5012 1092.72  5033.3 1092.96
  5061.9 1096.47  5119.2 1094.58  5154.3 1099.81  5218.1 1102.78  5397.5 1103.06
    5498 1103.48  5622.9 1104.83  5680.2 1110.16  5786.2 1114.85  5786.3 1114.85
#Mann= 6 ,-1 , 0
  4310.6     .07       0  4992.7     .05       0    5012     .07       0
  5397.5    .035       0    5498     .07       0  5786.2    .035       0
Bank Sta=4992.7,5012
XS Rating Curve= 0 ,0
Exp/Cntr=0.3,0.1

Type RM Length L Ch R = 1 ,70216   ,456,456,456
BEGIN DESCRIPTION:
West Fork 117.0
END DESCRIPTION:
XS GIS Cut Line= 3
      2185575.04       13822975.        2185375.       13822975.
      2184174.98     13822374.99
#Sta/Elev= 30
    4800 1147.86    4830  1144.8    4840 1141.59    4850 1137.99    4890  1120.2
    4920 1102.14    4940 1094.53    4950 1092.05  4960.4 1090.89  4960.9 1090.39
  4979.7 1090.89  4996.3 1091.18  5030.8  1093.6  5125.8 1092.81  5156.6 1094.18
  5192.9 1093.56  5237.6 1095.32    5260 1097.62  5313.1 1100.72  5504.4 1102.48
  5665.6 1102.16  5773.9 1103.44  5872.1 1105.64  5953.2 1111.89  6073.4 1115.42
  6113.5 1117.73  6148.7 1119.81  6221.5 1124.53  6288.6 1131.61  6341.7  1133.6
#Mann= 9 ,-1 , 0
    4800     .12       0  4960.4    .035       0  4979.7     .12       0
  4996.3    .035       0  5504.4     .07       0  5665.6    .035       0
  5773.9     .07       0  6113.5    .035       0  6148.7     .07       0
Bank Sta=4960.4,4979.7
XS Rating Curve= 0 ,0
Exp/Cntr=0.3,0.1

Type RM Length L Ch R = 1 ,69760   ,455,455,455
BEGIN DESCRIPTION:
West Fork 116.0
END DESCRIPTION:
XS GIS Cut Line= 3
      2185724.98       13822575.        2185525.       13822575.
      2185024.99       13822725.
#Sta/Elev= 30
  4804.6 1158.14  4834.6 1155.22  4844.6 1153.17  4854.6 1147.37  4884.6 1127.32
  4904.6 1110.45  4924.6 1096.45    4939 1089.55  4943.4 1087.74  4954.6 1084.02
  4964.6  1081.9  4964.9  1080.8  4965.4  1080.3  4984.2  1080.8  4994.6 1084.21
  5002.1  1085.8  5054.2 1089.44  5059.4 1088.93  5067.2 1090.51  5087.2 1092.61
  5119.4 1093.82  5125.5 1094.76  5130.7 1094.41  5158.6 1096.45  5163.8 1095.99
  5191.6 1098.04  5196.9 1097.54  5246.1  1098.8  5327.6 1098.38  5526.6 1101.88
#Mann= 7 ,-1 , 0
  4804.6     .12       0    4939     .07       0  4943.4    .035       0
  4964.9    .035       0  4984.2    .035       0  5246.1     .07       0
  5327.6    .035       0
Bank Sta=4964.9,4984.2
XS Rating Curve= 0 ,0
Exp/Cntr=0.3,0.1

Type RM Length L Ch R = 1 ,69305   ,466,466,466
BEGIN DESCRIPTION:
West Fork 115.0
END DESCRIPTION:
XS GIS Cut Line= 3
      2185824.99       13822175.        2185625.       13822175.
      2185074.97     13822575.02
#Sta/Elev= 30
  4800.1  1158.2  4810.1 1158.02  4820.1 1156.49  4860.1 1152.65  4880.1 1148.31
  4890.1 1142.59  4900.1 1135.17  4940.1  1111.9  4960.1 1099.75  4970.1 1092.84
  4980.1 1087.08  4987.9 1079.09  4988.4 1078.59  5006.7 1078.59  5007.2 1079.09
  5028.3 1079.88  5036.8  1080.6  5042.6 1080.34  5049.5  1083.4  5057.7 1084.99
  5099.4 1086.85  5136.1 1089.59    5179 1091.66  5193.7 1094.08  5204.2 1094.53
  5210.1  1094.8  5294.1 1096.05  5378.5 1096.12  5576.4 1098.05  5680.2 1099.41
#Mann= 8 ,-1 , 0
  4800.1     .12       0  4987.9     .05       0  5007.2     .12       0
  5028.3    .035       0  5204.2     .07       0  5210.1    .035       0
  5378.5     .07       0  5576.4    .035       0
Bank Sta=4987.9,5007.2
XS Rating Curve= 0 ,0
Exp/Cntr=0.3,0.1

Type RM Length L Ch R = 1 ,68839   ,443,443,443
BEGIN DESCRIPTION:
West Fork 114.0
END DESCRIPTION:
XS GIS Cut Line= 3
      2185775.02     13821775.01        2185575.       13821725.
      2185024.97     13821875.01
#Sta/Elev= 30
  4793.5 1124.51  4796.1 1124.51  4811.6 1120.55  4816.7 1120.27  4824.4    1118
    4876 1110.65    4894 1105.78  4906.9 1104.44  4922.2 1101.34  4927.5 1099.81
  4935.3 1095.89  4940.4 1096.65  4948.1 1094.26  4958.4 1089.46  4968.8  1081.4
  4979.7 1077.15  4980.2 1076.65    4999 1077.15    5017 1082.24  5041.1 1085.18
  5082.6  1084.6  5144.8 1088.33  5196.6 1088.58    5245 1091.45  5265.4 1091.55
  5289.9 1089.59  5319.3 1090.14  5352.1    1092    5473 1096.09  5569.8 1097.82
#Mann= 5 ,-1 , 0
  4793.5     .12       0  4922.2     .07       0  4979.7     .05       0
    4999     .07       0  5265.4    .035       0
Bank Sta=4979.7,4999
XS Rating Curve= 0 ,0
Exp/Cntr=0.3,0.1

Type RM Length L Ch R = 1 ,68396   ,488,488,488
BEGIN DESCRIPTION:
West Fork 113.0
END DESCRIPTION:
XS GIS Cut Line= 3
      2185975.04     13821625.02        2185425.       13821325.
      2184824.97     13820824.98
#Sta/Elev= 30
  4381.6 1131.45  4471.3 1123.26  4529.7 1114.76  4574.8 1110.41  4596.6 1106.19
    4712 1093.72  4852.9 1087.76  4869.1 1084.14  4900.2 1082.77  4934.6 1081.36
  4962.6 1082.16  4985.4 1080.13  5058.3 1081.99  5099.9 1080.05  5107.7 1081.44
  5136.4  1082.3  5161.8 1079.46  5162.3 1078.96  5181.2 1079.46  5192.3 1082.96
  5206.6 1084.91  5268.4 1089.73  5554.4 1093.96  5603.6 1097.19    5633 1101.15
  5689.6 1105.73  5703.9 1107.72  5718.2    1112  5750.6 1114.59  5789.2 1119.08
#Mann= 8 ,-1 , 0
  4381.6     .07       0  4900.2    .035       0  5161.8    .035       0
  5181.2    .035       0  5268.4     .07       0  5554.4    .035       0
  5603.6     .07       0  5750.6    .035       0
Bank Sta=5161.8,5181.2
XS Rating Curve= 0 ,0
Exp/Cntr=0.3,0.1

Type RM Length L Ch R = 1 ,67908   ,446,446,446
BEGIN DESCRIPTION:
West Fork 112.0
END DESCRIPTION:
XS GIS Cut Line= 3
        2186025.       13821475.        2185425.       13820875.
      2184825.02     13820625.01
#Sta/Elev= 30
  4147.3 1119.86  4157.1 1119.23  4246.3 1111.74  4274.6 1107.56  4303.2 1105.27
  4319.1 1103.91  4359.4 1101.66  4444.3 1094.14  4601.1  1090.4    4729 1089.12
  4769.6 1088.21  4826.1 1083.33  4862.9 1082.12  4939.3 1078.62  5000.6  1073.5
  5001.1    1073  5020.3  1073.5  5028.3 1075.51  5034.3  1078.6  5039.7    1079
  5058.1 1089.47  5119.8 1090.42  5341.9  1093.2    5396 1096.99  5461.7 1105.19
  5477.4 1106.15  5501.2 1111.28    5525 1114.83  5559.7 1118.26  5645.8 1130.07
#Mann= 11 ,-1 , 0
  4147.3    .035       0  4157.1     .07       0  4303.2    .035       0
  4319.1     .07       0  4601.1    .035       0    4729     .07       0
  4862.9    .035       0  5000.6    .035       0  5020.3    .035       0
  5119.8     .07       0    5396    .035       0
Bank Sta=5000.6,5020.3
XS Rating Curve= 0 ,0
Exp/Cntr=0.3,0.1

Type RM Length L Ch R = 1 ,67462   ,452,452,452
BEGIN DESCRIPTION:
West Fork 111.0
END DESCRIPTION:
XS GIS Cut Line= 3
      2185975.02     13820975.03        2185575.       13820475.
      2184975.03       13820525.
#Sta/Elev= 30
  4359.6 1092.24  4422.1 1090.49  4480.5 1089.71  4538.1 1087.38  4587.8 1087.47
  4643.8 1085.56  4765.4 1083.84  4858.3 1080.21  4885.5 1077.24  4943.1 1074.95
  4970.5 1072.44  4982.9 1071.59  4983.4 1071.09  5002.1 1071.09  5002.6 1071.59
    5010  1073.8    5020 1079.59  5030.1 1083.71  5040.1 1086.63  5100.3  1088.5
  5170.5 1087.87  5231.9 1089.04  5341.1 1090.47  5423.9 1093.13  5471.6 1097.92
  5501.7 1103.18    5515 1104.73  5561.9 1108.55    5582 1112.73    5602 1115.63
#Mann= 7 ,-1 , 0
  4359.6    .035       0  4422.1     .07       0  4970.5    .035       0
  4982.9    .035       0  5002.6    .035       0  5231.9     .07       0
    5515    .035       0
Bank Sta=4982.9,5002.6
XS Rating Curve= 0 ,0
Exp/Cntr=0.3,0.1

Type RM Length L Ch R = 1 ,67010   ,420,420,420
BEGIN DESCRIPTION:
West Fork 110.0
END DESCRIPTION:
XS GIS Cut Line= 3
        2186125.     13821325.02        2185825.       13820125.
      2185675.01     13819575.04
#Sta/Elev= 30
  3754.9 1110.53  3769.9 1108.56  3868.3 1103.06  3979.1 1096.81  4003.5 1096.44
  4084.8 1093.33    4261 1091.02  4589.8 1085.75  4685.2 1081.62  4734.2 1080.75
  4775.4 1081.69  4899.1 1076.05  5033.8  1072.1  5034.3  1071.6  5053.6  1072.1
    5054 1073.49  5107.6 1073.88  5237.2 1078.79  5261.3 1080.66  5271.7 1081.68
  5282.1 1085.64  5301.1 1089.19  5311.4 1090.84  5323.5 1095.15  5344.3 1098.99
  5356.4 1103.08  5396.1 1112.06  5458.3 1120.64  5470.4 1123.67  5561.9 1133.32
#Mann= 10 ,-1 , 0
  3754.9     .07       0  3769.9    .035       0  3868.3     .07       0
  4003.5    .035       0    4261     .07       0  5033.8     .05       0
  5053.6     .07       0  5107.6    .035       0  5301.1     .12       0
  5470.4     .07       0
Bank Sta=5033.8,5053.6
XS Rating Curve= 0 ,0
Exp/Cntr=0.3,0.1

Type RM Length L Ch R = 1 ,66590   ,410,410,410
BEGIN DESCRIPTION:
West Fork 109.0
END DESCRIPTION:
XS GIS Cut Line= 3
      2187225.04     13820675.03        2186025.       13819775.
        2185825.       13819475.
#Sta/Elev= 30
  3495.5  1126.9  3523.7 1131.54  3545.5 1124.44  3644.4 1117.32  3688.3  1115.5
  3717.4 1109.65  3773.7 1108.69  3862.6 1101.74  4024.2 1096.07  4098.5 1093.39
  4207.6 1089.33  4218.9  1088.9  4466.6 1081.14  4617.4 1080.59  4659.1 1076.95
  4700.6 1081.89  4802.8 1082.97  4883.5 1076.91  4917.4 1072.87  5042.5 1073.05
    5089 1072.78  5101.3 1071.82  5101.8 1071.32  5121.1 1071.82  5132.3  1075.2
  5163.2 1076.83  5219.4 1106.81  5276.5  1126.3    5320 1135.32  5356.1 1139.28
#Mann= 15 ,-1 , 0
  3495.5    .035       0  3644.4     .07       0  3862.6    .035       0
  4024.2     .07       0  4098.5    .035       0  4207.6     .07       0
  4218.9    .035       0  4466.6     .07       0  4700.6     .12       0
  4883.5     .07       0  5042.5    .035       0    5089     .07       0
  5101.3     .05       0  5121.1     .07       0  5163.2     .12       0
Bank Sta=5101.3,5121.1
XS Rating Curve= 0 ,0
Exp/Cntr=0.3,0.1

Type RM Length L Ch R = 1 ,66180   ,615,615,615
BEGIN DESCRIPTION:
West Fork 108.0
END DESCRIPTION:
XS GIS Cut Line= 3
      2186724.97     13820074.97        2186225.       13819525.
      2186124.99     13819324.97
#Sta/Elev= 30
  4252.2 1089.01  4257.8 1088.79  4358.2 1085.12  4419.4 1083.11  4499.9 1079.48
  4556.1 1077.99  4570.8 1076.51  4698.1 1076.94  4733.6 1074.96    4762 1078.74
  4804.6 1079.31  4846.8 1076.45  4874.8 1067.22  4882.3 1066.44  4896.5 1070.29
  4925.1 1072.51  4966.4 1068.65  4988.4 1067.75  4999.5 1065.16    5000 1064.66
  5019.3 1065.16  5040.2 1074.33  5054.2 1082.65  5062.5 1089.69  5076.5 1096.09
  5115.7 1120.51  5121.2 1121.37  5188.3  1151.4  5196.7 1153.53  5219.1 1154.74
#Mann= 10 ,-1 , 0
  4252.2     .07       0  4257.8     .12       0  4358.2     .07       0
  4419.4     .12       0  4499.9     .07       0  4556.1     .12       0
  4925.1     .07       0  4966.4     .12       0  4999.5     .05       0
  5019.3     .12       0
Bank Sta=4999.5,5019.3
XS Rating Curve= 0 ,0
Exp/Cntr=0.3,0.1

Type RM Length L Ch R = 1 ,65565   ,599,599,599
BEGIN DESCRIPTION:
H21662
END DESCRIPTION:
XS GIS Cut Line= 3
      2187438.31       13820105.      2186678.74     13819247.77
      2186429.61     13819204.44
#Sta/Elev= 30
  4024.5 1109.23  4066.2 1105.99  4336.4 1095.08  4501.6  1090.5  4565.2 1086.01
  4593.6 1078.84  4627.2 1074.84  4756.7 1071.22  4812.8  1075.2  4886.1 1073.87
  4912.3  1073.2  4983.4 1061.99  4994.4 1061.88  4994.9 1061.38  5014.2 1061.88
  5024.3 1062.33  5053.6 1062.81  5082.1 1075.42  5089.6 1084.89  5096.3 1086.76
  5103.8 1094.16  5110.5 1095.28  5118.1 1099.88  5153.2 1107.64  5194.6 1112.55
    5265 1125.91  5276.9 1130.05  5325.9 1138.79  5376.6 1150.87  5422.7 1158.51
#Mann= 9 ,-1 , 0
  4024.5    .035       0  4066.2     .07       0  4336.4     .12       0
  4627.2     .07       0  4886.1     .12       0  4994.4     .05       0
  5014.2     .12       0  5024.3    .033       0  5194.6     .12       0
Bank Sta=4994.4,5014.2
XS Rating Curve= 0 ,0
Exp/Cntr=0.3,0.1

Type RM Length L Ch R = 1 ,64966   ,773,773,773
BEGIN DESCRIPTION:
H21661
END DESCRIPTION:
XS GIS Cut Line= 3
      2188100.21     13820029.05      2187242.98     13819139.26
      2186648.14     13819041.93
#Sta/Elev= 30
  3918.4    1134  4019.7 1126.42  4108.8 1122.09  4130.1 1118.21  4151.6 1117.78
  4186.7 1114.26  4246.9 1112.43  4387.6 1104.17  4540.2 1092.98  4582.7 1091.84
  4596.8 1088.85  4618.2 1074.54  4632.2 1069.64  4646.2 1067.19  4681.7  1065.2
  4702.8 1067.48  4839.9 1067.22  5011.1 1064.87  5011.6 1064.37  5030.9 1064.87
  5077.6 1066.29  5113.1  1072.2  5153.6 1073.14  5303.9 1075.67  5435.6 1081.67
    5537  1097.2  5638.3 1109.35  5705.4 1121.87  5729.5 1124.04  5756.7 1132.03
#Mann= 9 ,-1 , 0
  3918.4    .035       0  4019.7     .07       0  4151.6    .035       0
  4246.9     .07       0  4387.6     .12       0  4839.9     .07       0
  5011.1     .05       0  5030.9     .07       0  5153.6     .12       0
Bank Sta=5011.1,5030.9
XS Rating Curve= 0 ,0
Exp/Cntr=0.3,0.1

Type RM Length L Ch R = 1 ,64193   ,543,543,543
BEGIN DESCRIPTION:
West Fork 105.0
END DESCRIPTION:
XS GIS Cut Line= 3
        2188325.       13818925.        2187925.       13818925.
      2186774.99       13818975.
#Sta/Elev= 30
  4605.1  1098.2  4745.1 1093.44  4775.1 1090.92  4835.1 1090.73  4905.1  1086.4
  4925.1 1079.15  4955.1 1062.96  4984.8 1053.12  4985.3 1052.62  5005.5 1053.12
  5045.1 1058.79  5075.2 1064.62  5085.2 1065.45  5135.2 1065.76  5305.4 1069.97
  5315.4  1070.9  5345.4 1070.45  5375.5 1071.59  5475.5  1071.7  5525.6 1070.22
  5545.6 1068.52  5555.7 1069.19  5615.7 1072.31  5654.4 1072.87  5851.9 1076.82
  5885.9 1078.04    5956  1084.8    6006 1091.67  6046.1 1095.78  6156.2 1111.79
#Mann= 6 ,-1 , 0
  4605.1     .12       0  4984.8     .05       0  5005.5     .12       0
  5555.7     .07       0  5654.4    .035       0  5851.9     .07       0
Bank Sta=4984.8,5005.5
XS Rating Curve= 0 ,0
Exp/Cntr=0.3,0.1

Type RM Length L Ch R = 1 ,63650   ,550,550,550
BEGIN DESCRIPTION:
West Fork 104.0
END DESCRIPTION:
XS GIS Cut Line= 3
      2188325.01       13818625.        2187975.       13818425.
      2186375.01     13819074.99
#Sta/Elev= 30
  4596.9 1095.32  4905.7 1079.64  4919.4 1077.64  4948.9 1066.37  4970.5 1064.14
    4976 1055.03  4976.5 1054.53  4996.7 1055.03  5068.3 1058.36  5129.5 1066.48
  5306.6 1067.68    5421 1063.77  5520.8 1068.45  5729.6 1071.61  5955.9 1077.74
  5961.4 1078.02  6026.9 1081.49  6069.1 1086.23  6199.3  1099.8  6289.2 1109.95
  6313.3 1115.26  6372.3 1123.32    6391 1128.18  6449.9 1138.03  6458.6  1141.1
  6498.1 1148.97  6565.1 1156.76  6629.2 1160.76    6673 1165.69    6727 1166.36
#Mann= 8 ,-1 , 0
  4596.9     .12       0    4976     .05       0  4996.7     .12       0
  5955.9     .07       0  5961.4    .035       0  6069.1     .12       0
  6199.3     .07       0  6458.6     .12       0
Bank Sta=4976,4996.7
XS Rating Curve= 0 ,0
Exp/Cntr=0.3,0.1

Type RM Length L Ch R = 1 ,63100   ,563,563,563
BEGIN DESCRIPTION:
West Fork 103.0
END DESCRIPTION:
XS GIS Cut Line= 3
        2187825.     13817525.01        2187825.       13817925.
      2187025.01     13818624.99
#Sta/Elev= 30
  4600.3 1099.87  4730.3 1096.32  4880.3 1087.35  4920.3 1083.44  4930.3 1081.61
  4940.3 1075.09  4950.3 1070.69  4960.3 1064.52  4970.3 1061.39  4980.3  1056.6
  4987.4 1048.73  4987.9 1048.23  5008.2 1048.73  5021.6  1052.2  5042.5 1053.66
  5064.4 1058.78  5113.7 1061.73  5226.7 1063.58  5312.1 1062.74    5333 1061.32
    5369 1063.33  5446.9  1065.3  5524.7 1066.23  5572.3 1065.52  5706.8 1066.69
  5807.7 1069.32  5921.4 1074.36  5943.2 1074.51    5985 1077.84  6063.3 1080.37
#Mann= 6 ,-1 , 0
  4600.3     .12       0  4987.4     .05       0  5008.2     .12       0
  5572.3     .07       0  5706.8    .035       0  5807.7     .12       0
#XS Ineff= 2 , 0
       0                    5230       0    1075
Permanent Ineff=
       F       F
Bank Sta=4987.4,5008.2
XS Rating Curve= 0 ,0
Exp/Cntr=0.3,0.1

Type RM Length L Ch R = 1 ,62537   ,561,561,561
BEGIN DESCRIPTION:
West Fork 102.0
END DESCRIPTION:
XS GIS Cut Line= 3
      2187175.02     13817275.04        2187375.       13817625.
      2186674.99     13818425.01
#Sta/Elev= 30
  4597.4 1128.58  4670.1 1120.87  4685.9 1116.43  4750.7 1111.23  4788.1  1105.5
  4831.3 1102.55  4868.7 1096.44  4911.9 1093.73  4949.4 1087.22  4955.1  1087.6
  4965.2 1079.49    4971 1081.23  4977.4 1071.99  4986.8 1065.27  4992.5 1065.28
  4997.2 1046.23  4997.7 1045.73    5018 1046.23  5042.7 1050.08  5050.3 1053.43
  5120.5 1052.72  5128.1 1054.78  5163.2 1055.45  5220.2 1059.73  5247.5 1059.69
    5709 1062.72  5787.6 1066.47    5858 1075.29  6013.7 1083.59  6063.5 1087.87
#Mann= 5 ,-1 , 0
  4597.4     .12       0  4997.2     .05       0    5018     .12       0
  5247.5    .035       0  5787.6     .12       0
Bank Sta=4997.2,5018
XS Rating Curve= 0 ,0
Exp/Cntr=0.3,0.1

Type RM Length L Ch R = 1 ,61976   ,571,571,571
BEGIN DESCRIPTION:
West Fork 101.0
END DESCRIPTION:
XS GIS Cut Line= 3
      2187074.99     13817225.02        2186825.       13817675.
        2186575.     13818474.99
#Sta/Elev= 30
  4492.8 1132.49  4506.5 1131.12  4538.5 1125.72    4566 1120.37    4582 1116.13
  4618.6 1110.66  4641.5 1105.88  4647.2 1103.74  4712.4 1093.32  4734.2 1088.36
  4801.6  1077.9  4824.5 1072.43  4869.1 1054.16  4874.9 1053.93  4886.2 1049.89
  4886.7 1049.39    4907 1049.89  4950.4  1052.2    5039 1049.91  5056.3 1052.79
    5094 1056.97  5129.7 1058.21  5294.1 1058.62  5396.8 1060.29  5494.2 1063.04
  5538.3 1065.25  5564.4 1068.24  5591.6 1073.15    5720 1082.51  5845.7 1092.98
#Mann= 5 ,-1 , 0
  4492.8     .12       0  4886.2     .05       0    4907     .12       0
  5129.7    .035       0  5538.3     .12       0
Bank Sta=4886.2,4907
XS Rating Curve= 0 ,0
Exp/Cntr=0.3,0.1

Type RM Length L Ch R = 1 ,61405   ,524,524,524
BEGIN DESCRIPTION:
West Fork 100.0
END DESCRIPTION:
XS GIS Cut Line= 3
        2186925.       13817025.        2186275.       13817625.
        2186325.     13818375.04
#Sta/Elev= 30
  4115.4 1140.93    4165 1137.61  4320.4 1105.51  4405.4 1090.84    4427 1088.42
  4476.3 1078.76  4511.5 1074.01  4610.7 1067.08  4752.5 1061.13  4780.8 1057.37
  4787.6 1053.89  4794.3 1053.88  4801.8 1050.97  4826.5 1048.47    4827 1047.97
  4847.4 1048.47  4934.8 1051.09  4964.6  1051.3    5010 1048.82  5040.1 1050.72
  5060.3 1053.79  5160.4 1056.65  5180.4 1055.51  5264.7 1057.13  5390.9  1060.2
  5448.2 1065.18  5491.1 1071.98  5571.3  1075.7  5711.6 1087.31  5751.7 1088.48
#Mann= 8 ,-1 , 0
  4115.4     .12       0  4794.3     .07       0  4826.5    .035       0
  4847.4     .07       0  4934.8    .035       0  5060.3     .07       0
  5264.7    .035       0  5448.2     .12       0
Bank Sta=4826.5,4847.4
XS Rating Curve= 0 ,0
Exp/Cntr=0.3,0.1

Type RM Length L Ch R = 1 ,60881   ,579,579,579
BEGIN DESCRIPTION:
West Fork 99.0
END DESCRIPTION:
XS GIS Cut Line= 3
        2186625.       13816825.        2185825.       13817475.
      2185925.01     13818075.04
#Sta/Elev= 30
  3964.2 1124.85  4041.8 1117.97  4070.5 1112.93  4148.8 1106.87  4255.8 1094.16
  4305.4 1086.58  4383.7 1077.47  4454.1 1067.16  4589.9 1061.29  4746.5 1057.73
  4829.5 1053.29  4923.9 1048.76  4997.5 1047.57  5004.8 1046.43  5005.3 1045.93
  5025.7 1046.43  5065.9 1047.93  5083.7 1053.82  5087.4 1053.41    5218 1055.89
    5289 1055.35  5309.3 1056.58    5327  1055.2  5359.9 1055.61  5400.5 1057.71
  5421.4 1060.62    5441 1062.72  5461.3  1062.2  5491.7 1068.41  5603.3  1072.9
#Mann= 6 ,-1 , 0
  3964.2     .12       0  4829.5     .07       0  5004.8     .05       0
  5025.7     .07       0  5087.4    .035       0  5421.4     .12       0
Bank Sta=5004.8,5025.7
XS Rating Curve= 0 ,0
Exp/Cntr=0.3,0.1

Type RM Length L Ch R = 1 ,60302   ,545,545,545
BEGIN DESCRIPTION:
West Fork 98.0
END DESCRIPTION:
XS GIS Cut Line= 3
      2186075.04     13816824.97        2185275.       13817375.
      2185425.01     13818025.04
#Sta/Elev= 30
  4034.2 1086.53  4070.7  1085.1  4271.7 1073.45  4328.5 1067.01  4358.3 1065.11
  4400.2 1060.22    4430 1059.07    4451 1056.56  4500.4 1055.13  4738.1 1052.71
  4752.7 1053.55  4803.5 1050.83  4890.1 1048.94  4946.9 1046.21  4981.1 1045.93
  4981.6 1045.43  5002.1 1045.93  5046.1 1046.47  5066.6 1047.61  5128.2 1047.76
  5155.5 1050.35  5189.8 1050.98  5230.9 1057.17  5290.7 1061.25  5333.5 1061.76
  5436.1 1067.18  5466.9 1067.19  5477.2 1068.12  5538.7 1068.85  5672.2  1072.3
#Mann= 5 ,-1 , 0
  4034.2     .12       0  4500.4     .07       0  4981.1     .05       0
  5002.1     .07       0  5155.5     .12       0
Bank Sta=4981.1,5002.1
XS Rating Curve= 0 ,0
Exp/Cntr=0.3,0.1

Type RM Length L Ch R = 1 ,59757   ,553,553,553
BEGIN DESCRIPTION:
West Fork 97.0
END DESCRIPTION:
XS GIS Cut Line= 3
      2185674.99       13816825.        2184875.       13817075.
      2184075.01     13817874.99
#Sta/Elev= 30
  4166.5 1070.34  4252.9 1067.43  4415.7 1057.22  4488.6 1052.55  4555.7 1051.16
  4732.2 1052.46  4820.8 1050.79  4899.9 1046.15  4983.6 1038.72  4984.1 1038.22
  5004.8 1038.72  5018.8 1043.46  5047.1 1045.47  5075.4 1050.36  5098.5 1049.82
  5117.8 1049.36  5131.9 1051.85  5155.1 1052.71  5233.6 1053.99  5407.2 1058.09
  5457.2 1058.16  5598.6 1062.37  5638.9 1062.11  5703.1  1064.2  5853.2 1072.86
  5952.2 1088.16  6051.2 1106.75  6107.7 1113.71  6121.9 1118.02    6136 1119.93
#Mann= 11 ,-1 , 0
  4166.5     .12       0  4415.7     .07       0  4488.6     .12       0
  4983.6     .05       0  5004.8     .12       0  5098.5     .07       0
  5155.1    .035       0  5233.6     .07       0  5407.2    .035       0
  5638.9     .07       0  5703.1     .12       0
Bank Sta=4983.6,5004.8
XS Rating Curve= 0 ,0
Exp/Cntr=0.3,0.1

Type RM Length L Ch R = 1 ,59204   ,546,546,546
BEGIN DESCRIPTION:
West Fork 96.0
END DESCRIPTION:
XS GIS Cut Line= 3
      2186175.04       13816675.        2184625.       13816625.
      2183874.99       13816275.
#Sta/Elev= 30
  3454.1 1091.52  3834.3    1073  4119.6 1062.77  4523.6 1050.42  4557.5 1049.73
  4681.5  1048.9    4741 1048.38  4934.9 1043.17  4984.2 1039.48  4984.7 1038.98
  5005.6 1039.48  5013.6  1041.2  5038.6 1041.44  5059.3  1043.2  5064.8 1041.74
  5082.2  1044.5  5126.3 1046.82  5276.1 1047.53  5395.9 1051.63  5435.3 1054.42
  5447.1 1058.04  5479.5 1061.93  5501.5  1067.5  5565.5 1074.96    5630  1082.1
  5679.9 1092.26  5698.6 1095.39  5755.3 1109.83  5783.5  1113.1  5832.6 1117.03
#Mann= 12 ,-1 , 0
  3454.1     .12       0  4119.6     .07       0  4523.6     .12       0
  4557.5     .07       0  4681.5     .12       0    4741     .07       0
  4984.2    .035       0  5005.6     .07       0  5038.6     .07       0
  5565.5     .12       0  5679.9     .07       0  5783.5     .12       0
Bank Sta=4984.2,5005.6
XS Rating Curve= 0 ,0
Exp/Cntr=0.3,0.1

Type RM Length L Ch R = 1 ,58658   ,569,569,569
BEGIN DESCRIPTION:
West Fork 95.0
END DESCRIPTION:
XS GIS Cut Line= 3
      2186025.01       13816625.        2184475.       13816125.
      2184124.98     13815924.99
#Sta/Elev= 30
  3376.7 1083.76    3585 1071.93  3782.6 1065.02  3828.5 1062.08  4135.2 1053.96
  4721.7 1047.12    4765 1045.34  4780.8 1042.79  4791.8 1040.71  4805.7 1040.47
  4848.5 1042.58  4893.2 1041.99  4984.2 1037.51  4984.7 1037.01  5005.6 1037.51
  5028.4 1042.13  5056.5 1040.09  5078.1 1042.48  5099.7 1053.45  5115.5 1064.61
  5137.1 1074.43  5152.9 1085.48  5166.6 1092.21  5174.5 1097.88  5189.6 1104.36
  5196.1 1109.81  5224.2 1121.36  5260.9 1128.39  5282.5  1130.6  5408.5 1131.47
#Mann= 6 ,-1 , 0
  3376.7     .12       0  4135.2     .07       0  4780.8     .12       0
  4848.5     .07       0  4984.2     .05       0  5005.6     .12       0
Bank Sta=4984.2,5005.6
XS Rating Curve= 0 ,0
Exp/Cntr=0.3,0.1

Type RM Length L Ch R = 1 ,58089   ,541,541,541
BEGIN DESCRIPTION:
West Fork 94.0
END DESCRIPTION:
XS GIS Cut Line= 3
      2186225.03     13816575.02        2184675.       13815625.
      2184275.01       13815725.
#Sta/Elev= 30
    3182 1092.36  3522.5 1072.34  3722.3 1063.34  3944.4 1054.73  4229.5 1050.11
  4359.6  1048.3  4628.7 1044.11  4724.5 1044.15  4824.1 1043.55  4847.5 1042.15
  4882.7 1036.85  4938.4 1035.97  4976.8 1035.33  4986.4 1032.88  4986.9 1032.38
  5007.8 1032.88  5030.9 1035.19  5051.5 1040.77  5059.3 1049.45  5064.4 1044.49
  5100.5 1071.37  5105.7 1068.34  5113.4 1073.98  5141.7 1080.17  5146.9 1079.79
  5188.1 1086.54  5216.5 1093.16  5247.4 1096.47  5311.8 1107.25  5412.3 1110.19
#Mann= 8 ,-1 , 0
    3182     .12       0  3722.3     .07       0  4229.5    .035       0
  4359.6     .07       0  4724.5    .035       0  4938.4     .12       0
  4986.4     .05       0  5007.8     .12       0
Bank Sta=4986.4,5007.8
XS Rating Curve= 0 ,0
Exp/Cntr=0.3,0.1

Type RM Length L Ch R = 1 ,57548   ,584,584,584
BEGIN DESCRIPTION:
West Fork 93.0
END DESCRIPTION:
XS GIS Cut Line= 3
      2185825.03     13816025.03        2185025.       13815225.
      2184625.02       13815175.
#Sta/Elev= 30
  3873.4 1057.68  3915.9 1055.75  4014.9 1052.71  4193.7 1049.34  4353.3 1046.22
  4410.8 1044.82  4599.4 1043.16  4757.3 1042.38  4783.8  1041.6    4821 1040.21
  4863.4 1037.22  4891.7 1036.33    4920 1034.26  4948.2 1034.02  4962.4 1032.81
  5004.1 1030.75  5004.6 1030.25  5025.1 1030.25  5025.6 1030.75    5035 1034.12
  5047.6 1044.12  5075.4 1048.21  5128.3 1053.67  5135.8 1055.07  5166.1 1058.75
  5236.6 1066.45  5256.8 1067.75  5347.5 1075.98  5365.1 1077.13  5407.9 1078.37
#Mann= 7 ,-1 , 0
  3873.4    .035       0  4193.7     .07       0  4353.3    .035       0
  4599.4     .07       0  4783.8     .12       0  5004.1     .05       0
  5025.6     .12       0
Bank Sta=5004.1,5025.6
XS Rating Curve= 0 ,0
Exp/Cntr=0.3,0.1

Type RM Length L Ch R = 1 ,56964   ,591,591,591
BEGIN DESCRIPTION:
West Fork 92.0
END DESCRIPTION:
XS GIS Cut Line= 3
      2186225.03     13815625.03        2185425.       13814825.
      2184874.98       13814775.
#Sta/Elev= 30
  3873.4 1058.44  3940.2 1056.97    4010 1055.66  4050.1  1054.9    4128  1053.3
  4453.3 1043.52  4598.2 1041.32    4821 1037.99  4835.1 1037.43  4861.4 1034.76
  4877.5 1033.52  4900.4 1033.17  4934.1 1034.61  4965.7 1032.43  4966.2 1031.93
  4986.8 1031.93  4987.3 1032.43  4990.7 1033.13  4996.6 1033.14  5034.9 1033.25
  5075.1 1037.91  5125.3 1040.34  5165.5 1040.95  5255.8 1044.33    5306 1047.39
  5356.3 1051.41  5446.6 1056.39  5476.7 1057.29  5506.9 1059.42  5557.1 1061.32
#Mann= 10 ,-1 , 0
  3873.4    .035       0  3940.2     .07       0    4010    .035       0
  4050.1     .07       0  4598.2    .035       0  4861.4     .12       0
  4900.4    .035       0  4965.7     .05       0  4987.3    .035       0
  4996.6     .12       0
Bank Sta=4965.7,4987.3
XS Rating Curve= 0 ,0
Exp/Cntr=0.3,0.1

Type RM Length L Ch R = 1 ,56373   ,539,539,539
BEGIN DESCRIPTION:
West Fork 91.0
END DESCRIPTION:
XS GIS Cut Line= 3
      2186374.98     13815274.96        2185875.       13814475.
      2185624.99     13813824.98
#Sta/Elev= 30
  4056.7 1055.15  4107.4 1053.67    4151 1052.91  4238.9 1048.43  4441.7 1044.04
    4477 1044.18  4595.3  1042.6  4714.2 1040.49  4934.6 1035.39  4964.7 1033.58
  4998.8 1029.51  4999.3 1029.01  5020.6 1029.51  5045.1 1030.72  5085.8 1030.98
  5139.3 1033.61  5246.5 1036.05  5318.3 1034.49  5372.9 1036.54  5401.8  1038.2
  5408.3 1040.07  5417.9 1041.22  5462.9 1046.03  5482.2 1046.74  5542.2  1054.4
  5572.2 1055.98  5596.8 1059.38  5656.8 1062.39    5675 1065.28  5696.5 1066.53
#Mann= 8 ,-1 , 0
  4056.7     .07       0  4107.4    .035       0  4238.9     .07       0
    4477    .035       0  4595.3     .07       0  4714.2     .12       0
  4998.8     .05       0  5020.6     .12       0
Bank Sta=4998.8,5020.6
XS Rating Curve= 0 ,0
Exp/Cntr=0.3,0.1

Type RM Length L Ch R = 1 ,55834   ,564,564,564
BEGIN DESCRIPTION:
West Fork 90.0
END DESCRIPTION:
XS GIS Cut Line= 3
      2186624.99     13815574.98        2186125.       13814025.
        2185775.       13813725.
#Sta/Elev= 30
  3371.4 1064.25  3426.2 1062.78  3530.6 1059.54  3705.8 1053.53  3777.2 1049.94
  3958.2 1046.93  4052.7 1045.97  4285.5 1044.31  4422.6 1041.73  4562.1  1039.1
  4690.3 1037.96  4747.8 1036.72  4759.7 1035.57  4842.4 1034.28  4914.7 1030.64
  4919.9 1029.31    4952  1029.1  5002.8 1026.76  5003.3 1026.26  5024.6 1026.76
  5042.3 1027.23  5127.9 1034.58  5170.7 1031.81  5205.8 1032.79  5276.6 1042.23
    5298 1044.31  5382.5 1057.37  5418.7 1060.07  5439.6 1063.93    5461 1064.33
#Mann= 9 ,-1 , 0
  3371.4    .035       0  3426.2     .07       0  3530.6     .12       0
  3705.8     .07       0  3958.2    .035       0  4052.7     .07       0
  4422.6     .12       0  5002.8     .05       0  5024.6     .12       0
Bank Sta=5002.8,5024.6
XS Rating Curve= 0 ,0
Exp/Cntr=0.3,0.1

Type RM Length L Ch R = 1 ,55270   ,525,525,525
BEGIN DESCRIPTION:
West Fork 89.0
END DESCRIPTION:
XS GIS Cut Line= 3
      2187224.98     13814274.98        2186425.       13813575.
        2186075.       13813375.
#Sta/Elev= 30
  3932.4 1051.84  3974.6 1051.57  4017.3 1047.62  4229.9 1039.82  4407.4 1036.45
  4463.9 1032.51  4534.6 1030.45  4577.3 1027.69  4598.2 1027.59    4620 1029.74
  4697.8 1032.48  4796.5 1033.43  4861.1 1032.64  4896.2 1031.31  4938.9 1027.99
  4959.8 1023.43  4981.6 1022.88  4992.4 1020.48  4992.9 1019.98  5014.2 1020.48
  5018.4 1021.63  5046.5 1022.79  5062.3 1025.13  5083.9 1026.37  5111.3 1031.61
    5143 1035.36  5207.7 1045.81  5282.6 1051.48  5353.2 1060.21  5398.5 1062.07
#Mann= 3 ,-1 , 0
  3932.4     .12       0  4992.4     .05       0  5014.2     .12       0
Bank Sta=4992.4,5014.2
XS Rating Curve= 0 ,0
Exp/Cntr=0.3,0.1

Type RM Length L Ch R = 1 ,54745   ,587,587,587
BEGIN DESCRIPTION:
West Fork 88.0
END DESCRIPTION:
XS GIS Cut Line= 3
        2187575.       13813225.        2186775.       13813225.
      2186375.01       13813125.
#Sta/Elev= 30
  4191.5 1063.43  4231.5  1061.8  4261.5 1057.83  4321.5 1052.65  4391.5 1049.92
  4471.5 1044.03  4491.5 1041.21  4511.5 1036.75  4581.5 1030.06    4605 1026.38
  4631.5  1023.2  4651.5 1022.65  4671.5 1023.67  4721.5 1029.07  4771.5 1029.47
  4931.5 1023.08  4971.5 1022.81  4994.1 1021.87  4998.6 1020.46  4999.1 1019.96
  5020.4 1020.46  5084.3 1023.95  5107.6 1028.13  5138.4 1036.32    5208 1039.08
  5249.2 1042.59  5256.9 1044.25  5298.2  1046.2  5331.7  1050.2  5403.8  1052.7
#Mann= 5 ,-1 , 0
  4191.5     .07       0    4605     .12       0  4998.6     .05       0
  5020.4     .12       0  5107.6     .12       0
Bank Sta=4998.6,5020.4
XS Rating Curve= 0 ,0
Exp/Cntr=0.3,0.1

Type RM Length L Ch R = 1 ,54158   ,531,531,531
BEGIN DESCRIPTION:
West Fork 87.0
END DESCRIPTION:
XS GIS Cut Line= 3
      2187525.01     13812624.99        2187175.       13812825.
      2186424.98       13812975.
#Sta/Elev= 30
  4596.9 1076.13  4691.2 1069.47  4796.6 1057.56  4809.3 1055.05  4825.1  1048.5
  4830.9 1048.16  4846.7 1044.18  4852.5  1043.8  4861.8 1040.44  4868.3 1034.48
  4874.1 1034.27  4884.1 1027.96  4889.9 1027.28  4896.4 1019.19  4937.7  1018.5
  4938.2    1018  4960.1  1018.5  5033.4 1021.19  5071.4 1022.73  5122.4 1021.14
  5211.3 1023.92  5256.4  1027.4  5312.4 1029.53  5377.4 1029.89  5428.3 1032.62
  5499.7 1034.26  5520.1 1035.51  5540.5  1038.9  5713.9 1044.42  5764.9 1048.08
#Mann= 8 ,-1 , 0
  4596.9     .07       0  4796.6     .12       0  4937.7     .05       0
  4960.1     .12       0  5033.4     .07       0  5211.3     .12       0
  5256.4     .07       0  5312.4     .12       0
Bank Sta=4937.7,4960.1
XS Rating Curve= 0 ,0
Exp/Cntr=0.3,0.1

Type RM Length L Ch R = 1 ,53627   ,557,557,557
BEGIN DESCRIPTION:
West Fork 86.0
END DESCRIPTION:
XS GIS Cut Line= 3
      2187474.97     13812175.02        2187125.       13812375.
      2186324.98     13812975.02
#Sta/Elev= 30
  4592.2 1088.22  4637.5 1087.31  4700.2 1084.06  4718.1 1083.39  4739.7  1079.8
  4857.1 1070.84  4877.8 1067.35  4914.7  1062.2  4922.6 1058.25  4937.7 1046.06
  4944.2 1027.58  4949.9 1023.25  4965.8 1018.97  4981.2 1010.09  4981.7 1009.59
  5003.6 1010.09  5017.1 1015.52  5034.1  1017.5  5045.3 1017.35  5051.3 1019.03
  5067.1 1020.96  5123.4 1023.98  5303.3 1026.53  5452.6 1030.51  5558.8 1031.86
  5623.4 1035.33  5673.4 1036.35  5731.7 1041.81  5867.1 1044.69  5995.3 1053.34
#Mann= 8 ,-1 , 0
  4592.2     .12       0  4700.2     .07       0  4877.8     .12       0
  4981.2     .05       0  5003.6     .12       0  5034.1     .07       0
  5051.3    .035       0  5303.3     .12       0
Bank Sta=4981.2,5003.6
XS Rating Curve= 0 ,0
Exp/Cntr=0.3,0.1

Type RM Length L Ch R = 1 ,53070   ,587,587,587
BEGIN DESCRIPTION:
West Fork 85.0
END DESCRIPTION:
XS GIS Cut Line= 3
      2187224.99       13811925.        2186825.       13811925.
      2186324.99     13812725.01
#Sta/Elev= 30
  4594.6 1077.24  4764.6 1062.37  4884.6 1055.21  4964.6 1045.21  4974.6 1042.36
  4984.6 1036.84  4992.1 1025.57  4997.5 1025.57  5002.3 1016.83  5008.1 1012.15
  5012.3 1010.12  5012.8 1009.62  5034.7 1010.12  5045.5 1012.67  5065.9 1012.94
  5096.6 1015.96  5124.3 1015.48  5154.4 1017.62  5175.6 1021.53  5196.8 1023.11
  5248.7 1025.47  5281.8 1025.36  5321.8 1023.39  5475.5 1025.24  5547.1 1026.55
  5626.1 1030.59  5735.7 1032.87  5830.1 1037.36  5866.6  1040.8    5938 1043.72
#Mann= 7 ,-1 , 0
  4594.6     .12       0  5012.3     .05       0  5034.7     .12       0
  5045.5     .07       0  5065.9     .12       0  5281.8    .035       0
  5475.5     .12       0
Bank Sta=5012.3,5034.7
XS Rating Curve= 0 ,0
Exp/Cntr=0.3,0.1

Type RM Length L Ch R = 1 ,52483   ,542,542,542
BEGIN DESCRIPTION:
West Fork 84.0
END DESCRIPTION:
XS GIS Cut Line= 3
      2186324.99     13811174.96        2186375.       13811575.
      2185874.98     13812375.04
#Sta/Elev= 30
  4592.6 1077.59  4693.4 1067.34  4743.8 1060.55  4796.7 1056.96  4877.3 1048.79
  4941.5 1040.76    4958 1039.15  4965.5 1035.46  4975.6 1029.07  4985.7 1012.03
  4993.2 1009.07  4998.1 1008.77  4998.6 1008.27  5020.6 1008.77    5040 1010.77
  5076.5 1010.33  5114.7 1012.92  5192.1 1019.15  5228.6 1020.67  5292.3 1022.14
  5342.5 1021.47  5432.1 1021.23  5475.1 1017.84  5500.7 1018.93  5511.7 1020.65
  5570.3 1022.71  5715.1 1025.27  5794.7 1029.72  5858.4 1031.05  5939.2 1035.29
#Mann= 9 ,-1 , 0
  4592.6     .12       0  4941.5     .07       0  4998.1     .05       0
  5020.6     .07       0  5114.7     .12       0  5228.6    .035       0
  5342.5     .12       0  5500.7     .07       0  5570.3     .12       0
Bank Sta=4998.1,5020.6
XS Rating Curve= 0 ,0
Exp/Cntr=0.3,0.1

Type RM Length L Ch R = 1 ,51941   ,567,567,567
BEGIN DESCRIPTION:
West Fork 83.0
END DESCRIPTION:
XS GIS Cut Line= 3
      2186175.02     13811224.98        2185875.       13811525.
      2185625.01     13812324.96
#Sta/Elev= 30
  4576.2 1069.75  4675.2 1062.64  4774.2 1054.13  4823.7 1051.63  4859.1 1047.56
  4873.2 1045.02  4901.5 1042.41  4915.6 1039.35  4929.8 1028.69  4943.9 1014.33
  4958.1 1007.95  4999.7 1006.26  5000.2 1005.76  5022.2 1006.26  5042.4 1006.31
  5049.2 1008.07  5067.4 1009.21  5086.9 1010.77  5105.3 1014.56  5151.9  1018.3
    5217 1015.14  5240.4 1016.03    5287 1019.24  5335.7 1018.88  5449.8 1020.38
  5622.3 1025.12  5702.4 1029.69  5775.8 1031.05  5807.2 1034.15  5838.6 1035.36
#Mann= 7 ,-1 , 0
  4576.2     .12       0  4999.7     .05       0  5022.2     .12       0
  5067.4     .07       0    5217     .12       0  5240.4     .07       0
  5449.8     .12       0
Bank Sta=4999.7,5022.2
XS Rating Curve= 0 ,0
Exp/Cntr=0.3,0.1

Type RM Length L Ch R = 1 ,51374   ,547,547,547
BEGIN DESCRIPTION:
West Fork 82.0
END DESCRIPTION:
XS GIS Cut Line= 3
      2185575.01     13810724.97        2185325.       13811475.
      2184674.98     13812025.02
#Sta/Elev= 30
  4209.4  1073.7  4388.6 1056.52  4441.3 1053.03  4462.4 1049.05  4525.7 1045.52
  4557.3  1040.2  4725.9 1030.25  4820.8 1021.28  4852.4 1020.56  4870.4 1018.43
  4884.1 1016.78  4894.6 1011.69  4915.7 1008.29  4947.3 1005.27  4978.2 1004.78
  4978.7 1004.28  5000.8 1004.78  5056.6 1008.18  5099.4 1007.95  5113.7 1009.37
  5134.6 1015.22    5206 1017.87    5262 1016.05  5526.5 1015.02  5575.2 1015.53
  5589.5 1018.63  5616.9 1029.05  5653.2 1034.61  5823.5  1044.3  5851.5 1044.73
#Mann= 5 ,-1 , 0
  4209.4     .12       0  4870.4     .07       0  4978.2     .05       0
  5000.8     .07       0  5526.5     .12       0
Bank Sta=4978.2,5000.8
XS Rating Curve= 0 ,0
Exp/Cntr=0.3,0.1

Type RM Length L Ch R = 1 ,50827   ,558,558,558
BEGIN DESCRIPTION:
West Fork 81.0
END DESCRIPTION:
XS GIS Cut Line= 3
      2185524.97     13810625.04        2184825.       13811425.
      2184575.02     13811874.96
#Sta/Elev= 30
  3936.9 1078.13    4036 1072.06  4199.3 1055.59  4234.4 1048.67  4262.9 1047.26
  4354.9 1038.85  4411.9 1035.88  4432.8 1032.59  4567.5 1021.56  4670.1  1017.1
  4808.6 1008.85  4829.5 1009.51  4914.9 1006.72  4957.6 1007.71  4985.2  1006.4
  4985.7  1005.9  5007.8  1006.4  5057.1 1008.26  5079.9 1014.33  5089.1 1015.53
  5182.9 1014.94  5263.4 1012.06  5308.7 1013.02  5331.6 1015.12  5354.5 1023.01
  5376.2 1033.22    5398 1038.18  5447.2 1041.08  5479.2 1045.22  5514.6 1047.85
#Mann= 5 ,-1 , 0
  3936.9     .12       0  4670.1     .07       0  4985.2     .05       0
  5007.8     .07       0  5263.4     .12       0
Bank Sta=4985.2,5007.8
XS Rating Curve= 0 ,0
Exp/Cntr=0.3,0.1

Type RM Length L Ch R = 1 ,50269   ,536,536,536
BEGIN DESCRIPTION:
West Fork 80.0
END DESCRIPTION:
XS GIS Cut Line= 3
        2185175.       13810475.        2184375.       13811125.
      2184274.99     13811575.05
#Sta/Elev= 30
  3965.2 1060.36  4071.5  1051.7  4093.8 1047.56  4164.2 1041.45  4263.3 1035.77
  4327.2 1028.64  4405.5 1022.23    4463 1019.37  4491.7 1015.86  4548.4 1013.59
    4626  1012.1  4791.9 1012.13  4854.2 1010.69  4963.3 1005.28  4977.5 1003.04
    4978 1002.54  5000.1 1003.04  5057.4 1003.86  5098.4 1006.03  5107.4 1006.87
  5118.9 1010.01    5156 1012.19  5253.4 1010.13  5307.9 1010.47  5354.5 1011.86
    5384 1018.47  5395.5 1024.85  5426.2 1032.27  5432.6  1033.6    5457 1033.95
#Mann= 7 ,-1 , 0
  3965.2     .12       0  4548.4     .07       0  4791.9     .12       0
  4963.3     .07       0  4977.5     .05       0  5000.1     .07       0
  5307.9     .12       0
Bank Sta=4977.5,5000.1
XS Rating Curve= 0 ,0
Exp/Cntr=0.3,0.1

Type RM Length L Ch R = 1 ,49733   ,593,593,593
BEGIN DESCRIPTION:
West Fork 79.0
END DESCRIPTION:
XS GIS Cut Line= 3
      2184525.01     13810074.99        2183925.       13810875.
        2184025.     13811374.99
#Sta/Elev= 30
  3994.3 1038.11  4001.6 1036.87    4087 1032.57  4101.6 1030.89  4224.2 1022.07
  4307.9 1016.28  4357.9 1014.18    4387 1011.76  4623.3 1009.07  4680.8 1008.62
  4701.6 1009.62  4802.5 1008.51  4851.6 1007.67  4907.9 1004.73    4987 1002.03
  5003.4 1000.36  5003.9  999.86  5026.1 1000.36  5075.9 1003.59  5106.5  1007.8
  5116.7 1008.34  5218.7 1007.84  5290.1 1009.09  5320.6 1012.33  5330.8 1012.59
  5371.6 1019.49  5381.8 1019.66  5408.5 1022.46    5443 1025.48  5504.2 1027.52
#Mann= 7 ,-1 , 0
  3994.3     .12       0  4224.2     .07       0  4623.3     .12       0
  4802.5     .07       0  5003.4     .05       0  5026.1     .07       0
  5408.5     .12       0
Bank Sta=5003.4,5026.1
XS Rating Curve= 0 ,0
Exp/Cntr=0.3,0.1

Type RM Length L Ch R = 1 ,49140   ,543,543,543
BEGIN DESCRIPTION:
West Fork 78.0
END DESCRIPTION:
XS GIS Cut Line= 3
      2184275.02     13809724.98        2183475.       13810525.
      2183075.01       13810575.
#Sta/Elev= 30
  3868.8 1047.07  4066.8 1032.68  4109.2 1030.68    4180 1019.81  4222.4 1014.75
  4256.5 1012.47  4349.7 1009.53  4519.4 1006.88  4547.6 1007.28  4575.9 1004.21
  4590.1 1003.89  4632.5 1003.92  4687.5 1006.77  4706.2 1007.25  4745.6 1007.37
  4773.9 1005.44  4831.1 1004.97  4964.8  1001.9  4996.7 1000.37    5043 1000.72
  5069.3   999.8  5069.8   999.3  5092.3   999.8  5111.1    1008  5118.6 1009.94
  5152.9 1014.51  5171.5 1016.74    5232 1020.43  5272.3 1021.15  5403.3 1026.94
#Mann= 8 ,-1 , 0
  3868.8     .12       0  4256.5     .07       0  4687.5    .035       0
  4706.2     .07       0  4831.1    .035       0  5069.3    .035       0
  5092.3    .035       0  5152.9     .12       0
Bank Sta=5069.3,5092.3
XS Rating Curve= 0 ,0
Exp/Cntr=0.3,0.1

Type RM Length L Ch R = 1 ,48597   ,547,547,547
BEGIN DESCRIPTION:
West Fork 77.0
END DESCRIPTION:
XS GIS Cut Line= 3
      2183874.98     13809525.01        2183125.       13810175.
      2182724.95       13810175.
#Sta/Elev= 30
  4007.5 1039.05  4043.1  1035.8  4113.3  1033.4  4145.8 1030.64  4184.6 1028.11
  4198.8 1025.93    4206 1023.11  4219.7 1021.81  4241.6 1021.99  4276.7 1019.74
    4291 1017.39  4311.8 1010.57    4348 1007.87  4553.1 1005.25  4620.1 1002.92
  4652.8 1000.94  4737.3 1002.95    4745 1000.95  4773.5  999.34  4837.1 1001.25
  4879.8 1000.08  4929.2 1001.26  4984.4   998.9  4984.9   998.4  5008.9   998.9
    5060 1000.45    5220 1033.57    5260  1038.1    5310 1048.52    5400 1057.08
#Mann= 5 ,-1 , 0
  4007.5     .12       0  4145.8    .035       0  4620.1     .12       0
  4984.4     .05       0  5008.9     .12       0
Bank Sta=4984.4,5008.9
XS Rating Curve= 0 ,0
Exp/Cntr=0.3,0.1

Type RM Length L Ch R = 1 ,48050   ,561,561,561
BEGIN DESCRIPTION:
West Fork 76.0
END DESCRIPTION:
XS GIS Cut Line= 3
      2183575.04     13809524.98        2183075.       13809725.
      2182574.98     13809875.01
#Sta/Elev= 30
  4457.3 1024.36  4500.1 1021.85    4526 1018.96  4532.7 1019.63  4651.2 1006.61
  4672.8 1006.35  4711.8 1003.55  4780.5 1002.54  4834.3  998.34  4888.2 1000.87
  4932.6  999.25  4951.4  999.63  5000.1  996.61  5000.6  996.11  5024.6  996.61
  5027.2  997.78  5050.7  997.44  5083.7  999.15  5267.3 1001.19  5292.5  1007.2
  5298.6 1010.49  5319.5 1016.57  5325.6  1019.9  5371.7  1037.6  5396.9 1044.65
    5403 1048.64  5413.5 1051.62  5455.2 1057.79  5486.6  1064.7  5517.9 1068.25
#Mann= 4 ,-1 , 0
  4457.3    .035       0  4500.1     .12       0  5000.1     .05       0
  5024.6     .12       0
Bank Sta=5000.1,5024.6
XS Rating Curve= 0 ,0
Exp/Cntr=0.3,0.1
