--- Mill Creek.prj (project) ---

Proj Title=Mill Creek Base Level Engineering
Current Plan=p01
Default Exp/Contr=0.3,0.1
English Units
Geom File=g01
Flow File=f01
Plan File=p01
Y Axis Title=Elevation
X Axis Title(PF)=Main Channel Distance
X Axis Title(XS)=Station
BEGIN DESCRIPTION:
Mill Creek
END DESCRIPTION:
DSS Export Rating Curves= 0
DSS Export Rating Curve Sorted= 0
DSS Export Volume Flow Curves= 0
DXF OffsetX= 0
DXF OffsetY= 0
DXF ScaleX= 1
DXF ScaleY= 10

--- Mill Creek.p01 (plan) ---

Plan Title=Multiple Run
Program Version=4.10
Short Identifier=Multiple
Geom File=g01
Flow File=f01
Subcritical Flow
K Sum by GR= 0
Std Step Tol= 0.01
Critical Tol= 0.01
Num of Std Step Trials= 20
Max Error Tol= 0.3
Flow Tol Ratio= 0.001
Split Flow NTrial= 30
Split Flow Tol= 0.02
Split Flow Ratio= 0.02
Log Output Level= 0
Friction Slope Method= 1
Unsteady Friction Slope Method= 2
Unsteady Bridges Friction Slope Method= 1
Parabolic Critical Depth
Global Vel Dist= 1 , 1 , 1
Global Log Level= 0
CheckData=True
Encroach Param=-1 ,0,0, 0
BEGIN DESCRIPTION:
Multiple Run
END DESCRIPTION:
Computation Interval=1HOUR
Output Interval=1HOUR
Run HTab= 0
Run UNet= 0
Run PostProcess= 0
Run WQNet= 0
UNET Theta= 1
UNET Theta Warmup= 1
UNET ZTol= 0.02
UNET ZSATol= 0.05
UNET MxIter= 20
UNET MaxInSteps= 0
UNET DtIC= 0
UNET DtMin= 0
UNET MaxCRTS= 20
UNET WFStab= 2
UNET SFStab= 1
UNET WFX= 1
UNET SFX= 1
UNET DSS MLevel= 4
UNET DZMax Abort= 100
UNET Convert EG Bridges= 0
UNET Use Existing IB Tables=-1
UNET Froude Reduction=False
UNET Froude Limit= 1
UNET Froude Power= 10
UNET Time Slicing=0,0, 5
UNET Junction Losses=0
Instantaneous Interval=1HOUR
Write IC File= 0
Write IC File at Sim End=0
Echo Input=False
Echo Parameters=False
Echo Output=False
Write Detailed= 0
WQ AD Non Conservative
WQ ULTIMATE=-1
WQ Max Comp Step=1HOUR
WQ Output Interval=15MIN
WQ Output Selected Increments= 0
WQ Output face flow=0
WQ Output face velocity=0
WQ Output face area=0
WQ Output face dispersion=0
WQ Output cell volume=0
WQ Output cell surface area=0
WQ Output cell continuity=0
WQ Output cumulative cell continuity=0
WQ Output face conc=0
WQ Output face dconc_dx=0
WQ Output face courant=0
WQ Output face peclet=0
WQ Output face adv mass=0
WQ Output face disp mass=0
WQ Output cell mass=0
WQ Output cell source sink temp=0
WQ Output cell source sink nsm=0
WQ Output MaxMinRange=-1
WQ Daily Max Min Mean=-1
WQ Daily Range=0
WQ Daily Time=0
WQ Create Restart=0
WQ Fixed Restart=0
WQ System Summary=0
WQ Use Fixed Temperature=0
Sorting and Armoring Iterations= 10
XS Update Threshold= 0.02
Hydraulics Update Threshold= 0.02
Energy Slope Method= 1
Volume Change Method= 0
XS Weighting Method= 0
Number of US Weighted Cross Sections= 1
Number of DS Weighted Cross Sections= 1
Upstream XS Weight=0.25
Main XS Weight=0.5
Downstream XS Weight=0.25
Number of DS XS's Weighted with US Boundary= 1
Upstream Boundary Weight= 1
Weight of XSs Associated with US Boundary= 0
Number of US XS's Weighted with DS Boundary= 1
Downstream Boundary Weight= 0.5
Weight of XSs Associated with DS Boundary= 0.5
Sediment Output Level= 4
Mass or Volume Output= 0
Output Increment Type= 1
Profile and TS Output Increment= 10
XS Output Flag= 0
XS Output Increment= 10
Disregard all LS=0
Disregard all Conn=0
Disregard all Breaches=0
Disregard all Pumps=0

--- Mill Creek.f01 (steady flow) ---

Flow Title=Multiple
Number of Profiles=7
Profile Names=10-year,25-year,50-year,1pct_min,100-year,1pct_plu,500-year
River Rch & RM= Mill Creek,Reach-1,97478
     896    1498    2061    1375    2743    5473    4813
River Rch & RM= Mill Creek,Reach-1,96354
    1306    2224    3098    2088    4166    8313    7471
River Rch & RM= Mill Creek,Reach-1,93039
    1425    2430    3389    2285    4559    9097    8183
River Rch & RM= Mill Creek,Reach-1,88561
    1482    2530    3530    2381    4751    9480    8537
River Rch & RM= Mill Creek,Reach-1,87278
    1525    2596    3614    2431    4850    9678    8666
River Rch & RM= Mill Creek,Reach-1,83718
    1614    2735    3796    2543    5073   10123    8992
River Rch & RM= Mill Creek,Reach-1,70963
    2770    4791    6740    4568    9115   18187   16542
River Rch & RM= Mill Creek,Reach-1,61991
    3880    6790    9630    6575   13119   26177   24156
River Rch & RM= Mill Creek,Reach-1,58673
    4176    7293   10328    7038   14042   28018   25751
River Rch & RM= Mill Creek,Reach-1,50416
    4455    7786   11030    7517   14998   29926   27512
River Rch & RM= Mill Creek,Reach-1,47688
    4569    7990   11325    7721   15406   30739   28281
River Rch & RM= Mill Creek,Reach-1,47116
    4745    8293   11749    8005   15972   31869   29281
River Rch & RM= Mill Creek,Reach-1,41154
    4791    8364   11839    8059   16081   32085   29426
River Rch & RM= Mill Creek,Reach-1,36942
    5542    9698   13749    9371   18697   37305   34288
River Rch & RM= Mill Creek,Reach-1,30874
    5625    9839   13947    9503   18961   37833   34756
River Rch & RM= Mill Creek,Reach-1,25265
    5548    9688   13714    9332   18620   37151   34036
River Rch & RM= Mill Creek,Reach-1,22051
    6098   10640   15056   10237   20425   40753   37272
River Rch & RM= Mill Creek,Reach-1,15263
    6169   10740   15176   10302   20555   41012   37387
River Rch & RM= Mill Creek,Reach-1,2616
    6109   10623   14997   10171   20294   40491   36845
Boundary for River Rch & Prof#=Mill Creek,Reach-1,1
Up Type=0
Dn Type=3
Dn Slope=0.0009
Boundary for River Rch & Prof#=Mill Creek,Reach-1,2
Up Type=0
Dn Type=3
Dn Slope=0.0009
Boundary for River Rch & Prof#=Mill Creek,Reach-1,3
Up Type=0
Dn Type=3
Dn Slope=0.0009
Boundary for River Rch & Prof#=Mill Creek,Reach-1,4
Up Type=0
Dn Type=3
Dn Slope=0.0009
Boundary for River Rch & Prof#=Mill Creek,Reach-1,5
Up Type=0
Dn Type=3
Dn Slope=0.0009
Boundary for River Rch & Prof#=Mill Creek,Reach-1,6
Up Type=0
Dn Type=3
Dn Slope=0.0009
Boundary for River Rch & Prof#=Mill Creek,Reach-1,7
Up Type=0
Dn Type=3
Dn Slope=0.0009

--- Mill Creek.g01 (geometry) ---

Geom Title=Existing Conditions
Program Version=4.10

River Reach=Mill Creek      ,Reach-1
Reach XY= 30
        2325075.       13793275.      2328622.95     13792019.14
      2327581.87     13788474.88      2328424.51     13787909.78
      2327582.08     13786974.99      2328174.64     13783690.16
      2326276.62     13780318.99       2326919.3     13778922.46
      2325191.48     13778542.06      2324469.61     13775522.56
        2322975.       13774425.      2322328.53     13769976.45
      2323122.57     13768680.52      2329234.69     13765764.25
      2330122.55     13764030.47       2330984.8     13764564.53
      2331772.57     13762580.52      2333991.83     13763109.47
      2334968.79      13759282.8      2336973.45     13759921.25
      2337318.95     13758132.45      2340849.48     13757152.17
      2339525.08     13754109.61      2339841.27     13752657.77
        2340475.       13753025.      2339428.46      13751776.5
      2340744.96     13751905.84      2342918.66     13748533.02
      2343126.48     13749421.55        2343925.       13748925.

Type RM Length L Ch R = 1 ,97478   ,359,359,359
BEGIN DESCRIPTION:
B19456
END DESCRIPTION:
XS GIS Cut Line= 3
      2325188.18     13794015.25      2325129.62     13793266.95
      2324668.81     13792715.28
#Sta/Elev= 30
  4297.2  641.21  4368.9  637.71  4432.6  636.03  4540.3  632.54  4588.3  631.57
  4650.1  628.05  4795.2  621.74    4819  620.26  4829.1  620.69  4859.2     619
  4943.8  617.03  4989.6  615.51  5007.6  610.12  5007.9  609.62  5011.6  610.12
  5046.3  613.25  5123.6  612.95  5222.5  615.52  5279.8  614.15  5407.3  617.66
  5450.3  619.95  5456.8  621.17  5499.7  624.63    5557  627.13  5612.9  631.06
  5649.4  632.39  5662.7  633.99  5684.5  634.77  5727.5  639.67  5766.6  642.31
#Mann= 9 ,-1 , 0
  4297.2    .035       0  4368.9     .07       0  4432.6    .035       0
  4540.3     .07       0  4650.1     .12       0  4795.2     .07       0
  4943.8     .12       0  5007.6     .05       0  5011.6     .12       0
Bank Sta=5007.6,5011.6
XS Rating Curve= 0 ,0
Exp/Cntr=0.3,0.1

Type RM Length L Ch R = 1 ,97119   ,765,765,765
BEGIN DESCRIPTION:
Mill Creek 131.0
END DESCRIPTION:
XS GIS Cut Line= 3
        2325825.       13793775.        2325325.       13793075.
      2324925.01     13792675.01
#Sta/Elev= 30
  4144.4  626.24  4208.3  625.06  4237.8  623.32  4267.3  620.83  4296.8  616.45
  4316.4  615.33  4344.7  615.98  4409.8  613.58  4466.4  615.36  4567.1  614.98
  4581.9  614.13  4644.3  613.62  4660.5   614.1  4724.4  612.52  4750.1  610.71
  4783.4  609.11  4825.2   608.9  4890.3   611.2  4918.6  610.82  4955.5  609.34
  4965.8  607.31    4966  606.81  4969.8  607.31  4991.1  607.43  4997.3  608.84
  5018.8  610.66  5117.8  610.49  5372.3  617.58  5428.9  621.67  5570.3  627.75
#Mann= 6 ,-1 , 0
  4144.4     .07       0  4296.8     .12       0  4644.3     .07       0
  4750.1     .12       0  4965.8     .05       0  4969.8     .12       0
Bank Sta=4965.8,4969.8
XS Rating Curve= 0 ,0
Exp/Cntr=0.3,0.1

Type RM Length L Ch R = 1 ,96354   ,886,886,886
BEGIN DESCRIPTION:
B19455
END DESCRIPTION:
XS GIS Cut Line= 5
      2326287.92     13793963.26      2325963.49     13793220.03
      2325805.46     13793078.83      2325585.12     13792876.52
      2324675.32     13792259.15
#Sta/Elev= 30
  4195.4  623.44  4297.1  621.16  4463.5  618.64  4614.4  614.64  4880.9  611.85
  4940.5  613.34  4963.9  606.53  4992.8  605.22  5008.7   607.2  5013.9  605.09
  5014.2  604.59  5018.5  605.09  5037.1  607.65    5058  606.33  5243.5  606.09
  5494.2  609.04  5532.3  609.39  5541.3  611.57  5547.3  609.65  5562.2  613.28
  5604.2  614.89  5634.1  613.11  5855.5  617.27  5894.7  617.67  5942.6   619.1
  6023.4  616.89  6140.7  619.87  6255.5  624.13  6475.6  638.88  6616.9  641.85
#Mann= 12 ,-1 , 0
  4195.4     .07       0  4297.1    .035       0  4463.5     .07       0
  5013.9     .05       0  5018.5     .07       0    5058    .035       0
  5243.5     .07       0  5494.2    .035       0  5855.5     .12       0
  5894.7    .035       0  6140.7     .12       0  6255.5     .07       0
Bank Sta=5013.9,5018.5
XS Rating Curve= 0 ,0
Exp/Cntr=0.3,0.1

Type RM Length L Ch R = 1 ,95468   ,603,603,603
BEGIN DESCRIPTION:
B19454
END DESCRIPTION:
XS GIS Cut Line= 4
      2326424.55     13793449.17      2326418.04     13793188.86
      2326157.75     13792824.46      2325676.19     13792271.31
#Sta/Elev= 30
  4486.2  615.15  4530.4  620.34  4610.4  622.44  4640.4  619.36  4666.8   614.1
  4671.8  615.86  4740.4  604.05  4841.8   602.8  4965.4  601.83  4993.8  597.82
  4994.1  597.32  4998.5  597.82    5017  602.44  5031.8  602.54  5037.9  605.59
  5046.3  602.27  5067.4  602.73  5073.5  604.23  5082.1  603.05  5088.3  604.53
  5095.4  603.22  5119.3  603.49  5298.5  605.05  5394.1  606.23  5472.1  609.42
  5615.7  620.12  5634.3  620.85  5883.5  640.76  5924.5  644.45  5927.8  644.48
#Mann= 11 ,-1 , 0
  4486.2    .035       0  4841.8     .12       0  4965.4      .1       0
  4993.8     .05       0  4998.5      .1       0  5119.3     .12       0
  5298.5    .035       0  5615.7     .12       0  5634.3    .035       0
  5883.5     .12       0  5924.5    .035       0
Bank Sta=4993.8,4998.5
XS Rating Curve= 0 ,0
Exp/Cntr=0.3,0.1

Type RM Length L Ch R = 1 ,94865   ,475,475,475
BEGIN DESCRIPTION:
Mill Creek 126.0
END DESCRIPTION:
XS GIS Cut Line= 3
      2326474.97     13793425.04        2326825.       13793025.
      2326124.98     13792274.98
#Sta/Elev= 30
    4469  621.95    4497   623.2  4511.3  621.46  4582.5  605.31  4589.1   606.5
  4675.6  604.73  4824.3  602.07  4887.1  601.13  4915.6  598.71  4936.5  598.68
  4950.7  597.82  4958.3  594.83  4970.2  594.67  4970.5  594.17    4975  594.67
  4986.8  596.44  4993.4  595.53  4997.2  597.31  5014.5  598.72  5085.8  599.47
  5163.5  600.17  5241.2  598.84  5413.7  600.49  5651.5  602.39  5785.9  605.52
  5842.5  611.17  5915.5  622.98  5934.4  626.04  5984.2  637.91  6026.5  641.76
#Mann= 8 ,-1 , 0
    4469    .035       0  4675.6     .07       0  4824.3     .12       0
  4970.2     .05       0    4975     .12       0  5085.8      .1       0
  5413.7     .12       0  5915.5    .035       0
Bank Sta=4970.2,4975
XS Rating Curve= 0 ,0
Exp/Cntr=0.3,0.1

Type RM Length L Ch R = 1 ,94390   ,445,445,445
BEGIN DESCRIPTION:
Mill Creek 125.0
END DESCRIPTION:
XS GIS Cut Line= 3
        2327375.       13793575.        2327175.       13792775.
        2326375.       13792125.
#Sta/Elev= 30
  4183.3  621.93  4296.7  616.55  4337.9  610.76  4390.8  605.98    4490  602.66
  4712.9  599.33  4736.1  598.82  4769.9   597.8  4838.3  596.53  4925.5  595.15
  4940.5  591.77  4966.7   592.1  4984.7  589.15  4989.9  591.01  4995.2  589.06
  4995.6  588.56    5000  589.06  5005.3  591.61  5015.1  590.84  5021.6  595.67
  5050.7  595.64  5114.2  594.12  5157.3  595.86  5526.5  598.33  5775.8  604.39
  5818.9  607.61  5874.9   614.7  5903.7  615.78  5967.6  625.05  6038.7  629.52
#Mann= 10 ,-1 , 0
  4183.3     .07       0  4390.8    .035       0  4712.9     .07       0
  4736.1     .12       0  4769.9     .07       0  4838.3     .12       0
  4940.5      .1       0  4995.2     .05       0    5000      .1       0
  5050.7    .035       0
Bank Sta=4995.2,5000
XS Rating Curve= 0 ,0
Exp/Cntr=0.3,0.1

Type RM Length L Ch R = 1 ,93945   ,464,464,464
BEGIN DESCRIPTION:
Mill Creek 124.0
END DESCRIPTION:
XS GIS Cut Line= 3
        2327525.     13793575.04        2327575.       13792825.
        2326775.       13792075.
#Sta/Elev= 30
  4248.8  623.12  4271.4  621.36    4319  617.13    4339  617.11  4399.2  612.71
  4459.3  607.56    4501  606.63    4590  602.09    4777  597.39  4875.4  595.72
  4950.4   594.3  5026.2  589.18  5026.5  588.68  5031.1  589.18  5056.9  592.54
  5108.8  593.71  5163.3  593.34  5184.4  590.09  5205.9  590.72  5212.7  592.61
  5226.9   591.2  5233.8  593.33  5345.2  593.69  5623.1  594.59  5870.7  597.23
  5998.2  600.88  6026.5  602.87  6040.7  606.51  6075.8  607.63  6097.1  609.61
#Mann= 11 ,-1 , 0
  4248.8     .07       0  4271.4    .035       0    4501     .07       0
    4590     .12       0    4777     .07       0  4875.4     .12       0
  5026.2     .05       0  5031.1     .12       0  5108.8      .1       0
  5163.3     .12       0  5345.2    .035       0
Bank Sta=5026.2,5031.1
XS Rating Curve= 0 ,0
Exp/Cntr=0.3,0.1

Type RM Length L Ch R = 1 ,93481   ,442,442,442
BEGIN DESCRIPTION:
Mill Creek 123.0
END DESCRIPTION:
XS GIS Cut Line= 3
      2328175.04     13792725.02        2327925.       13792575.
      2327124.99     13791824.99
#Sta/Elev= 30
    4709  599.86    4849  595.76  4949.6  589.88  4965.6  589.84  4989.8  583.94
  4990.3  583.44  4995.8  583.94    5004  584.01  5007.7   587.6  5021.8  589.47
    5142  588.29  5276.3  589.23  5304.7  585.72    5312   589.4  5318.7  589.15
  5381.6  590.45  5458.8  590.43  5545.5  592.84  5644.4  593.16  5755.9   595.2
  5770.7  595.64  5807.3  596.85  5884.9  603.07  5891.8  604.85  5941.6  609.62
  5948.5  611.72  5976.8  615.31  6005.1  617.67  6061.8  621.85  6097.2  622.78
#Mann= 10 ,-1 , 0
    4709     .12       0  4949.6      .1       0  4989.8     .05       0
  4995.8      .1       0  5318.7     .12       0  5381.6      .1       0
  5458.8    .035       0  5644.4     .07       0  5755.9    .035       0
  5770.7     .07       0
Bank Sta=4989.8,4995.8
XS Rating Curve= 0 ,0
Exp/Cntr=0.3,0.1

Type RM Length L Ch R = 1 ,93039   ,472,472,472
BEGIN DESCRIPTION:
Mill Creek 122.0
END DESCRIPTION:
XS GIS Cut Line= 3
        2328275.     13792574.99        2328125.       13792225.
        2327475.       13791825.
#Sta/Elev= 30
  4618.7  599.54  4727.5  595.11  4856.2  588.02  4918.8  586.09  4932.4  585.16
  4966.8  586.74  4990.4  585.05  5004.1  582.61  5004.6  582.11  5010.2  582.61
  5013.1  584.76  5043.9  586.29  5058.2  583.27  5065.2  583.92    5071  586.21
  5116.9  585.85  5123.1  583.58  5144.4  584.92  5152.1  586.37  5165.4  586.36
  5196.5  586.33  5202.4  584.06  5223.7  586.88  5291.2  589.63  5358.4  590.23
  5398.7  591.03  5486.3  596.11  5507.7  598.59  5645.3  608.18  5762.7  612.23
#Mann= 7 ,-1 , 0
  4618.7     .12       0  4918.8      .1       0  5004.1     .05       0
  5010.2      .1       0  5165.4     .12       0  5358.4    .035       0
  5486.3     .07       0
Bank Sta=5004.1,5010.2
XS Rating Curve= 0 ,0
Exp/Cntr=0.3,0.1

Type RM Length L Ch R = 1 ,92567   ,493,493,493
BEGIN DESCRIPTION:
B19453
END DESCRIPTION:
XS GIS Cut Line= 3
      2329046.96     13792668.31      2328259.57     13791939.49
      2327128.69     13791471.53
#Sta/Elev= 30
  4246.2  628.23  4440.8   617.4    4519  611.19  4631.8  605.23    4646   603.2
  4822.9  598.57  4950.5   596.8  4957.4  595.35  4971.5  588.42  4978.8  584.89
    4993  581.86  4999.8  578.22  5004.1   577.5  5004.6     577  5010.3   577.5
  5028.2  583.48  5035.5  583.76  5219.2  585.63  5264.7  585.01  5400.7  582.89
  5518.9  586.88  5655.4  589.19  5738.5  589.79  5883.7  598.69  5993.7  604.13
  6067.6  604.95  6214.6  604.35  6366.8  606.55  6384.7  608.21    6543  611.16
#Mann= 10 ,-1 , 0
  4246.2     .12       0  4971.5      .1       0  5004.1     .05       0
  5010.3      .1       0  5264.7     .12       0  5655.4    .035       0
  5883.7     .07       0  6067.6    .035       0  6214.6     .07       0
  6366.8    .035       0
Bank Sta=5004.1,5010.3
XS Rating Curve= 0 ,0
Exp/Cntr=0.3,0.1

Type RM Length L Ch R = 1 ,92074   ,409,409,409
BEGIN DESCRIPTION:
B19452
END DESCRIPTION:
XS GIS Cut Line= 4
      2329463.41     13792342.94       2328832.2     13791763.79
      2328148.95     13791757.28      2326899.79     13791230.29
#Sta/Elev= 30
  3821.9  622.65  3830.1  622.11  3968.2  618.03  4078.9  612.59  4218.7  605.75
  4300.5  601.79  4477.3  597.26  4735.7  591.69  4775.7  588.02  4805.7  581.27
  4886.9  582.53  4965.8  582.29  5002.7  577.42  5003.2  576.92  5008.9  577.42
  5025.8  581.08  5065.8  582.26  5215.9  581.78  5275.8  582.09    5446  586.36
  5640.4  588.37  5702.6   593.4  5857.3  598.38    5988  598.72  6076.1  597.67
  6178.3  600.22  6258.3  601.89    6459  606.73  6505.7  606.44  6717.6  615.27
#Mann= 14 ,-1 , 0
  3821.9     .12       0  3830.1     .07       0  4078.9     .12       0
  4218.7     .07       0  4477.3     .12       0  4886.9      .1       0
  5002.7     .05       0  5008.9      .1       0  5215.9     .12       0
    5446    .035       0  5857.3     .07       0    5988    .035       0
  6178.3     .07       0  6258.3    .035       0
Bank Sta=5002.7,5008.9
XS Rating Curve= 0 ,0
Exp/Cntr=0.3,0.1

Type RM Length L Ch R = 1 ,91665   ,452,452,452
BEGIN DESCRIPTION:
B19451
END DESCRIPTION:
XS GIS Cut Line= 4
      2329411.31     13792128.17      2328584.93     13791340.82
      2328148.95     13791477.48      2327055.78     13791087.06
#Sta/Elev= 30
  3545.1   612.2  3826.7  601.88  4001.7  597.26  4073.8  595.67  4138.9  594.29
  4307.4  591.72    4413  590.71  4882.7  579.59  4926.7  580.07  4958.9  579.87
  4976.5  572.73    4977  572.23  4982.8  572.73  5000.8  579.99  5011.3  580.39
  5063.7  578.69  5164.6  583.04  5492.7  587.73  5523.5  590.53  5529.9  593.68
    5549     591  5554.3   593.6  5572.9  589.63  5677.8  594.52  5711.5  596.35
  5764.5  599.73  5874.4  600.68    6122  606.25  6126.2  606.35  6304.2   611.8
#Mann= 17 ,-1 , 0
  3545.1     .12       0  3826.7     .07       0  4001.7     .12       0
  4073.8     .07       0  4138.9     .12       0  4307.4      .1       0
    4413     .12       0  4882.7      .1       0  4926.7    .035       0
  4976.5    .035       0  4982.8    .035       0  5572.9     .07       0
  5677.8    .035       0  5711.5     .07       0  5874.4    .035       0
    6122     .07       0  6126.2    .035       0
Bank Sta=4976.5,4982.8
XS Rating Curve= 0 ,0
Exp/Cntr=0.3,0.1

Type RM Length L Ch R = 1 ,91213   ,574,574,574
BEGIN DESCRIPTION:
B19450
END DESCRIPTION:
XS GIS Cut Line= 3
       2329378.8     13792030.58      2328435.27     13791119.58
      2327270.49     13790833.27
#Sta/Elev= 30
  3420.7  608.06  3639.1  600.76  3730.5  598.68  4116.6  591.31  4347.9  588.53
  4466.7  586.76  4514.3  587.16  4587.7  587.44  4594.1  588.44  4664.9  585.93
  4700.4  582.32  4797.4  578.47  4936.6  578.07  4959.1     576  4980.1  572.02
  4980.6  571.52  4986.5  572.02    4990  573.49  5031.2  577.46  5061.3   576.2
  5066.4  573.85  5082.6  575.45  5113.5  575.55  5141.5  578.73  5216.5  581.66
  5388.3  583.87  5570.1   589.9  5703.2  599.98  5888.9  609.26  5931.7  610.16
#Mann= 15 ,-1 , 0
  3420.7     .12       0  3639.1     .07       0  3730.5     .12       0
  4116.6      .1       0  4347.9     .12       0  4466.7      .1       0
  4514.3     .12       0  4587.7    .035       0  4797.4     .12       0
  4980.1     .05       0  4986.5     .12       0  5141.5     .07       0
  5388.3    .035       0  5703.2     .07       0  5888.9    .035       0
Bank Sta=4980.1,4986.5
XS Rating Curve= 0 ,0
Exp/Cntr=0.3,0.1

Type RM Length L Ch R = 1 ,90639   ,523,523,523
BEGIN DESCRIPTION:
B19449
END DESCRIPTION:
XS GIS Cut Line= 4
      2329697.64     13791197.66      2328441.77     13790852.79
      2328155.46     13790696.61      2327349.29     13790586.09
#Sta/Elev= 30
  3619.4  604.62  3668.8   602.8  4006.3   592.3  4206.3  589.99  4316.9  588.79
    4348  585.87  4404.3   585.7  4438.8  591.91  4462.1  592.37  4478.4  591.42
  4493.2  586.68  4580.7  582.57  4648.8  576.93  4690.6  577.22    4785   579.4
  4919.3   577.9  4963.6  576.77    4975  575.01  4994.6   568.5  4995.1     568
  5001.1   568.5  5007.3  572.18  5020.6  573.69  5088.9   576.3  5329.1   575.8
  5379.6  578.68  5446.9  579.69    5666  583.15  6005.4  604.15  6061.6  605.11
#Mann= 10 ,-1 , 0
  3619.4     .07       0  3668.8     .12       0  4006.3     .07       0
  4206.3     .12       0  4580.7    .035       0  4690.6     .07       0
  4919.3     .12       0  4994.6     .05       0  5001.1     .12       0
  5446.9     .07       0
Bank Sta=4994.6,5001.1
XS Rating Curve= 0 ,0
Exp/Cntr=0.3,0.1

Type RM Length L Ch R = 1 ,90116   ,351,351,351
BEGIN DESCRIPTION:
B19448
END DESCRIPTION:
XS GIS Cut Line= 3
      2329652.15     13790599.01      2328493.83     13790462.36
      2327491.72     13790488.38
#Sta/Elev= 30
  4098.9  597.37  4158.1  594.88  4245.8  593.56  4267.2  591.43    4388  588.34
  4613.6  585.72  4730.4  585.21  4818.1  583.18  4931.8  581.06  4940.4  580.61
  4951.9  576.09  4957.4  576.13    4962  576.17  4972.1   579.3  4982.1  576.74
  4992.2  570.07  4998.9  567.83  4999.4  567.33  5005.7  567.83  5022.4  572.42
  5052.6  574.09  5143.2  572.12  5193.6  573.17  5213.7  571.88  5466.8  574.36
  5622.4  575.72  5905.7  578.87  5964.3  581.28  6014.3  587.06  6267.7  598.81
#Mann= 11 ,-1 , 0
  4098.9     .07       0  4158.1     .12       0  4245.8     .07       0
  4613.6    .035       0  4818.1     .07       0  4957.4     .12       0
  4998.9     .05       0  5005.7     .12       0  5466.8     .07       0
  5622.4     .12       0  5905.7     .07       0
Bank Sta=4998.9,5005.7
XS Rating Curve= 0 ,0
Exp/Cntr=0.3,0.1

Type RM Length L Ch R = 1 ,89765   ,365,365,365
BEGIN DESCRIPTION:
B19447
END DESCRIPTION:
XS GIS Cut Line= 3
      2329554.53     13790462.37      2328695.55     13790189.05
      2327550.28     13790423.32
#Sta/Elev= 30
  4008.2  591.73  4180.9  587.64    4329  585.34  4439.1  585.78  4490.4  583.27
  4572.9  582.76  4584.9  581.92  4603.7  582.49  4771.1  581.79  4868.2  582.89
  4889.2  582.77  4910.9  581.41  4914.8  581.51  4930.6  576.14    4951  570.96
  4971.4   569.7  4978.2  564.62  4978.7  564.12  4985.1  564.62  5010.6  570.91
  5167.1  571.36    5196  570.65    5254  571.65  5409.3  575.35    5517   576.5
  5712.1  576.94  5790.5  578.14    5813  578.73  5951.3  589.78  6078.6  595.52
#Mann= 11 ,-1 , 0
  4008.2     .07       0    4329    .035       0  4439.1     .07       0
  4603.7     .12       0  4771.1     .07       0  4910.9     .12       0
  4978.2     .05       0  4985.1     .12       0    5254     .07       0
    5517     .12       0  5790.5     .07       0
Bank Sta=4978.2,4985.1
XS Rating Curve= 0 ,0
Exp/Cntr=0.3,0.1

Type RM Length L Ch R = 1 ,89400   ,382,382,382
BEGIN DESCRIPTION:
B19446
END DESCRIPTION:
XS GIS Cut Line= 4
      2329495.94     13790351.74      2328676.03     13789935.27
      2328279.09     13790006.85      2327512.58     13790370.62
#Sta/Elev= 30
  3743.3  588.96  3980.9  585.32  3981.4  585.31  4032.3   586.4  4082.4  583.23
  4142.1   582.7  4307.9  581.23  4446.7  581.06  4510.5  581.44  4583.1  581.27
  4634.5  579.31    4666  574.78  4689.5  569.64  4714.8  568.39  4836.7  569.33
  4855.3  566.46  4877.3  569.33  4948.5  569.75  4969.1  563.73  4969.6  563.23
    4976  563.73  4999.3  569.78  5047.9  569.47  5148.7  573.89  5238.9  574.45
  5573.7  576.83  5637.1  578.32  5705.3  583.31  5779.2  590.91  5914.7  596.79
#Mann= 13 ,-1 , 0
  3743.3     .07       0  3980.9    .035       0  3981.4     .07       0
  4142.1     .12       0  4307.9     .07       0  4446.7     .12       0
  4510.5     .07       0  4634.5     .12       0  4969.1     .05       0
    4976     .12       0  5047.9     .07       0  5238.9     .12       0
  5573.7     .07       0
Bank Sta=4969.1,4976
XS Rating Curve= 0 ,0
Exp/Cntr=0.3,0.1

Type RM Length L Ch R = 1 ,89018   ,457,457,457
BEGIN DESCRIPTION:
B19445
END DESCRIPTION:
XS GIS Cut Line= 4
      2329404.81      13790241.1      2328610.96     13789707.52
      2328038.33     13789759.58       2327563.3      13790228.1
#Sta/Elev= 30
  3555.2  587.01    3627  585.99  3698.3  586.88  3719.9  585.29  3790.1   582.8
  4047.4  580.18  4095.7  579.56  4154.6  579.28  4396.5  578.06  4402.1  578.48
  4417.1  574.47  4453.1  569.08  4768.7  566.86  4982.7  568.17  5006.2  562.27
  5006.7  561.77  5013.2  562.27  5039.8  568.51  5059.9  566.18    5080  568.61
  5149.4  567.61  5156.5  569.54  5163.6  567.83  5170.7  569.96  5194.3  570.12
  5401.8  576.12  5516.2  577.95    5602  580.15  5644.4  585.15  5753.9  591.19
#Mann= 13 ,-1 , 0
  3555.2     .07       0    3627    .035       0  3698.3     .07       0
  3719.9     .12       0  4047.4     .07       0  4095.7     .12       0
  4154.6     .07       0  4396.5     .12       0  5006.2     .05       0
  5013.2     .12       0  5194.3     .07       0  5401.8     .12       0
  5516.2     .07       0
Bank Sta=5006.2,5013.2
XS Rating Curve= 0 ,0
Exp/Cntr=0.3,0.1

Type RM Length L Ch R = 1 ,88561   ,369,369,369
BEGIN DESCRIPTION:
Mill Creek 113.0
END DESCRIPTION:
XS GIS Cut Line= 3
      2328674.97     13789574.99        2328025.       13789325.
        2327625.       13789525.
#Sta/Elev= 30
  4295.1  575.83  4354.2  575.11  4389.4   569.5  4402.2  568.31    4474  567.67
  4487.9  568.42  4605.8  566.18  4672.9  566.61  4704.5  566.36  4734.3  564.46
  4766.5  565.72  4812.6  562.86  4820.1   565.2  4837.2  566.23  4861.8  566.56
  4891.8  565.05  4927.2   564.5  4946.5  565.69  4994.3  565.66  4999.9  565.33
  5010.2  558.49  5010.7  557.99  5017.5  558.49  5022.2  559.89  5027.8  563.99
  5036.2  565.61  5111.7  564.78  5171.6   567.9  5223.5  570.11  5438.7  574.81
#Mann= 7 ,-1 , 0
  4295.1     .12       0  4354.2    .035       0  4672.9     .07       0
  4704.5     .12       0  5010.2     .05       0  5017.5     .12       0
  5171.6     .07       0
Bank Sta=5010.2,5017.5
XS Rating Curve= 0 ,0
Exp/Cntr=0.3,0.1

Type RM Length L Ch R = 1 ,88192   ,381,381,381
BEGIN DESCRIPTION:
B19444
END DESCRIPTION:
XS GIS Cut Line= 3
      2329001.41     13789252.03      2327908.18     13789011.26
      2327179.67       13789356.
#Sta/Elev= 30
  3732.4  577.21    3743  577.53  3769.7  574.25  3788.1   575.2  3884.4  574.25
  4083.4  570.18  4128.1  568.89  4230.5  570.06  4350.4  567.45  4355.7  567.11
  4676.3  564.13  4844.9  561.64  4898.5   563.3  4925.5  563.12  4954.9   563.5
  4973.4  559.51  4973.9  559.01  4980.7  559.51  4985.9  562.89  4991.4  563.51
  5021.2  560.17  5043.4  564.36  5105.2  568.58  5165.1  568.57  5173.4  567.13
  5275.8  571.09  5353.2  570.81    5452  572.88  5586.6  581.41  5657.8  586.39
#Mann= 13 ,-1 , 0
  3732.4     .12       0  3788.1    .035       0  3884.4     .07       0
  4083.4     .12       0  4350.4     .07       0  4355.7     .12       0
  4676.3      .1       0  4898.5     .12       0  4925.5      .1       0
  4973.4     .05       0  4980.7      .1       0  5021.2     .12       0
  5586.6    .035       0
Bank Sta=4973.4,4980.7
XS Rating Curve= 0 ,0
Exp/Cntr=0.3,0.1

Type RM Length L Ch R = 1 ,87811   ,533,533,533
BEGIN DESCRIPTION:
B19443
END DESCRIPTION:
XS GIS Cut Line= 3
      2328923.35     13789076.34      2327771.53     13788744.46
      2327108.88     13788685.99
#Sta/Elev= 30
  3754.9   578.3  3783.9   576.9  3878.1  573.76  3923.6  573.75  3957.2  571.29
  4013.3  570.15  4029.8  570.92  4063.5  568.93  4138.2  568.08  4190.3  565.33
  4208.5  566.56  4281.1  566.66  4596.1  564.73  4700.2  560.89  4762.6  561.06
  4788.9  559.84  4908.3  562.27  4990.2  562.42  4999.8  560.58  5004.8   561.5
  5010.3   557.8  5016.7  557.32  5017.2  556.82  5024.1  557.32  5040.4  561.41
  5080.6  562.24  5140.8  566.06  5291.4  569.76  5472.1  577.75  5618.8  580.45
#Mann= 5 ,-1 , 0
  3754.9    .035       0  3783.9     .07       0  4138.2     .12       0
  5016.7     .05       0  5024.1     .12       0
Bank Sta=5016.7,5024.1
XS Rating Curve= 0 ,0
Exp/Cntr=0.3,0.1

Type RM Length L Ch R = 1 ,87278   ,653,653,653
BEGIN DESCRIPTION:
B19442
END DESCRIPTION:
XS GIS Cut Line= 4
       2328890.8     13789004.76      2327927.71     13788568.77
       2327556.8     13788165.32      2326932.13     13787937.58
#Sta/Elev= 30
  3697.9  578.18  3879.7  571.81  3974.8  568.92    4104  565.36  4141.9  564.83
  4154.3  563.05  4216.7  564.94  4417.9  564.71  4593.4  558.73  4631.3  559.03
  4637.3  556.72  4659.9   559.4  4704.1  559.86  4858.5  558.94  4964.6  560.72
  4982.3  553.79  4982.8  553.29  4990.2  553.79    4993  556.02  5000.4  555.88
  5014.6  559.34    5042   560.7    5079  561.52  5127.4  564.49  5210.9  565.47
  5251.2  566.19  5509.3  569.61  5567.2  569.96  5856.9     571    5968  575.09
#Mann= 15 ,-1 , 0
  3697.9     .07       0  3879.7     .12       0  3974.8     .07       0
    4104     .12       0  4704.1      .1       0  4858.5     .12       0
  4982.3     .05       0  4990.2     .12       0    5042      .1       0
    5079     .12       0  5210.9     .07       0  5251.2     .12       0
  5509.3     .07       0  5567.2     .12       0  5856.9    .035       0
Bank Sta=4982.3,4990.2
XS Rating Curve= 0 ,0
Exp/Cntr=0.3,0.1

Type RM Length L Ch R = 1 ,86625   ,422,422,422
BEGIN DESCRIPTION:
B19441
END DESCRIPTION:
XS GIS Cut Line= 3
      2328903.76     13788646.84      2327875.65     13788204.37
      2326978.79     13787885.92
#Sta/Elev= 30
  4315.5  583.57  4499.2  574.73  4536.3  574.58  4659.4  568.57  4784.6  565.26
  4934.6  556.92    4940  558.09  4956.5  556.66    4969  553.62  4978.2  555.52
  4992.5  555.71    5041  552.51  5041.5  552.01  5049.2  552.51  5054.5  557.81
  5076.7  558.14  5197.1  557.48  5215.2  555.39  5244.2  557.88  5261.3  556.68
  5283.1  558.29  5320.3  557.93  5444.3  562.29  5763.5  566.38    6058  568.97
  6138.2  567.73  6256.3  569.51  6287.2  568.27  6309.3  569.85  6386.5  572.88
#Mann= 9 ,-1 , 0
  4315.5     .07       0  4784.6     .12       0    5041     .05       0
  5049.2     .12       0  5076.7      .1       0  5320.3     .12       0
  5763.5     .07       0    6058     .12       0  6309.3    .035       0
Bank Sta=5041,5049.2
XS Rating Curve= 0 ,0
Exp/Cntr=0.3,0.1

Type RM Length L Ch R = 1 ,86203   ,589,589,589
BEGIN DESCRIPTION:
B19440
END DESCRIPTION:
XS GIS Cut Line= 3
      2328936.28     13788093.74      2327498.23     13787905.04
       2326899.8     13787813.97
#Sta/Elev= 30
  4430.9  584.22  4458.5  582.54  4512.9     583  4543.1   581.1  4654.1  578.82
  4810.1  572.27  4909.1  567.71  4921.1  567.21  4956.7  556.68  4994.8  553.82
  4995.7  547.28  4996.2  546.78  5003.9  547.28  5007.1  550.08  5017.2  553.86
  5057.5  550.48  5067.6  555.61  5072.6   555.9  5167.9  554.88  5198.7  553.11
  5231.1  553.81  5289.5  557.82  5462.4  559.02  5853.3  564.27  5975.6  566.08
  6126.8  565.88  6181.8  565.02  6317.5  569.56  6469.2  575.67  6486.6  576.07
#Mann= 10 ,-1 , 0
  4430.9    .035       0  4810.1     .07       0  4909.1      .1       0
  4995.7     .05       0  5003.9      .1       0  5167.9     .12       0
  5853.3     .07       0  6126.8     .12       0  6317.5    .035       0
  6469.2     .07       0
Bank Sta=4995.7,5003.9
XS Rating Curve= 0 ,0
Exp/Cntr=0.3,0.1

Type RM Length L Ch R = 1 ,85614   ,674,674,674
BEGIN DESCRIPTION:
B19439
END DESCRIPTION:
XS GIS Cut Line= 3
      2328806.17     13787605.71      2328298.61     13787605.71
      2326893.02     13787755.38
#Sta/Elev= 30
  4519.1  575.87  4610.3  574.34    4849  562.71  4900.3  559.39  4930.3  554.43
  4950.3  553.73  4976.1  547.13  4976.6  546.63  4984.4  547.13  5000.3  552.78
  5048.1  553.71  5080.6  551.56  5110.7  552.75  5130.9  550.11  5158.8  553.04
  5246.5  552.31  5446.3  554.84  5533.1  553.86  5778.6  560.87  5918.8  561.95
  5995.7  559.57  6016.3  561.48    6046  561.32  6086.2  565.17  6217.2  567.09
  6242.8  567.92  6337.6  572.41  6347.7  571.28    6397  573.43  6440.2  574.68
#Mann= 10 ,-1 , 0
  4519.1     .07       0    4849    .035       0  4976.1    .035       0
  4984.4    .035       0  5048.1      .1       0  5246.5     .12       0
  5778.6     .07       0  6217.2     .12       0  6242.8    .035       0
    6397     .07       0
Bank Sta=4976.1,4984.4
XS Rating Curve= 0 ,0
Exp/Cntr=0.3,0.1

Type RM Length L Ch R = 1 ,84940   ,344,344,344
BEGIN DESCRIPTION:
B19438
END DESCRIPTION:
XS GIS Cut Line= 3
      2328552.39     13787456.04      2327966.75      13787332.4
      2326951.66     13787638.23
#Sta/Elev= 30
  4213.3   565.5  4294.2  561.59  4547.9  555.82  4577.4  553.77  4878.7  549.65
  4959.9  549.99  4976.2  547.56  4977.3  544.53  4977.8  544.03  4985.6  544.53
  5009.2  545.45  5047.4  554.09  5081.3  554.91  5137.4  556.92  5262.8  557.68
  5288.9  557.01  5321.8  551.97  5346.3  555.49  5387.8  558.19  5393.1  557.05
    5409  558.94  5431.3  558.44  5440.3  559.52  5459.1  567.87  5471.6   566.9
  5492.1  562.28  5576.1  562.26    5608   564.1  5852.8  571.28    5872   571.3
#Mann= 7 ,-1 , 0
  4213.3     .07       0  4878.7    .035       0  4977.3    .035       0
  4985.6    .035       0  5081.3     .07       0    5608    .035       0
  5852.8     .07       0
Bank Sta=4977.3,4985.6
XS Rating Curve= 0 ,0
Exp/Cntr=0.3,0.1

Type RM Length L Ch R = 1 ,84596   ,322,322,322
BEGIN DESCRIPTION:
B19437
END DESCRIPTION:
XS GIS Cut Line= 3
      2328604.48     13787443.03        2327739.     13787111.16
      2326710.89     13787169.72
#Sta/Elev= 30
  4010.8  565.98  4138.8  561.85  4310.1  558.64    4351  556.69  4381.1  557.13
  4405.7  555.29  4435.5  555.15  4674.3  550.13  4920.6  547.57  4975.6  545.07
  4997.6  543.35  4998.1  542.85    5006  543.35  5041.9   546.2  5071.9  551.08
  5090.1  552.82  5164.5  556.53  5182.1  558.18  5212.2  557.89  5275.1   560.7
  5366.2   562.5  5370.6  562.68  5471.2  563.78  5495.8  563.57    5733  566.74
  5763.1   567.6  5783.1  570.18  5797.3  568.08  5893.3  571.63  5967.5  572.79
#Mann= 11 ,-1 , 0
  4010.8     .07       0  4435.5     .05       0  4975.6     .07       0
  4997.6     .05       0    5006     .07       0  5164.5     .05       0
  5275.1     .07       0  5366.2     .12       0  5370.6     .07       0
  5471.2     .05       0  5495.8     .07       0
Bank Sta=4997.6,5006
XS Rating Curve= 0 ,0
Exp/Cntr=0.3,0.1

Type RM Length L Ch R = 1 ,84274   ,556,556,556
BEGIN DESCRIPTION:
B19436
END DESCRIPTION:
XS GIS Cut Line= 3
        2328624.     13787417.01      2327517.75     13786772.79
      2326802.67     13786499.75
#Sta/Elev= 30
  3909.2  567.19  3993.6  563.57  4208.9  557.97  4232.1  558.45  4347.8   556.1
  4362.7   556.7  4451.9  553.41  4458.7  554.34  4623.6  549.81  4822.7  547.68
  4854.1  548.38  4891.4  546.81  4903.2  544.43  4912.9  544.21  4934.4  546.64
  4961.7   546.6  4971.6  546.16  4988.9  542.24  4989.4  541.74  4997.3  542.24
  5007.4  543.31  5014.6  551.12  5030.3  554.28    5181  555.07  5252.2  557.96
  5352.9  558.88  5394.1  560.22  5778.1  562.51  5840.9  563.33  5954.8  562.81
#Mann= 7 ,-1 , 0
  3909.2     .07       0  3993.6     .05       0  4623.6     .12       0
  4988.9     .05       0  4997.3     .12       0  5394.1     .07       0
  5778.1     .12       0
Bank Sta=4988.9,4997.3
XS Rating Curve= 0 ,0
Exp/Cntr=0.3,0.1

Type RM Length L Ch R = 1 ,83718   ,477,477,477
BEGIN DESCRIPTION:
B19435
END DESCRIPTION:
XS GIS Cut Line= 3
      2328890.77     13787078.62      2328122.92     13786668.67
      2326932.13     13786336.81
#Sta/Elev= 30
  4129.7   565.6  4232.8  564.31  4306.3  561.71  4328.9  562.52    4431  558.45
  4453.6  559.17  4521.7  556.49  4660.5  554.47  4715.6  551.32  4816.4  548.74
  4978.4  547.72  4986.4  546.95  4994.7  542.17  4998.7  538.62  5004.1  538.23
  5004.6  537.73  5012.6  538.23  5033.4  544.57  5060.3  543.53  5101.8  546.24
  5217.9  544.38  5332.9  549.15  5350.9  548.96  5367.1  550.84  5480.1  551.91
    5652  556.68  5806.3  557.88    5819  557.14  6005.5  559.71  6236.3  560.51
#Mann= 6 ,-1 , 0
  4129.7     .07       0  4715.6     .12       0  5004.1     .05       0
  5012.6     .12       0  5217.9     .12       0  5806.3     .07       0
Bank Sta=5004.1,5012.6
XS Rating Curve= 0 ,0
Exp/Cntr=0.3,0.1

Type RM Length L Ch R = 1 ,83241   ,789,789,789
BEGIN DESCRIPTION:
B19434
END DESCRIPTION:
XS GIS Cut Line= 3
      2329001.36     13786492.97      2328201.01     13786258.72
      2327010.21     13786167.62
#Sta/Elev= 30
  4243.8  554.37  4615.3  550.19  4859.8  550.38  4872.3  549.12  4957.7  545.67
  4990.2  544.96  5006.8  535.65  5007.3  535.15  5015.3  535.65  5037.3  542.35
  5083.4   543.9  5123.9  542.65  5148.2  543.82    5271  542.44  5314.4  540.03
  5404.7  541.09  5484.9   539.4    5505  541.61  5535.1  548.26  5582.8  550.88
  5635.4   551.5  5658.2  547.44  5675.5  550.65  5705.6  552.28  5785.8  553.83
  5815.9     551  5835.9  552.65  5876.1  551.98  5914.2  555.53    6272  559.19
#Mann= 10 ,-1 , 0
  4243.8     .07       0  4872.3    .035       0  4957.7     .12       0
  5006.8     .05       0  5015.3     .12       0  5083.4      .1       0
  5148.2     .12       0    5271      .1       0  5658.2     .12       0
  5914.2     .07       0
Bank Sta=5006.8,5015.3
XS Rating Curve= 0 ,0
Exp/Cntr=0.3,0.1

Type RM Length L Ch R = 1 ,82452   ,512,512,512
BEGIN DESCRIPTION:
B19433
END DESCRIPTION:
XS GIS Cut Line= 3
      2328981.87     13785386.76      2328617.47     13785718.62
      2327128.71     13786082.69
#Sta/Elev= 30
  3691.5  551.38  3730.3  551.61  3744.5  552.63  3758.7   551.8  3886.4   552.6
  3921.5  552.16  4014.4  548.86  4169.5  544.61  4207.5  544.77    4259  543.44
  4413.4  544.72  4524.2  544.21  4619.3  544.97  4699.6  544.28  4856.1  541.74
    4959  538.04  4979.6  538.66  4987.4  538.36  4992.5  536.58  5006.1  535.84
  5006.6  535.34  5014.9  535.84  5051.7  542.59  5070.7  545.08  5097.3  546.03
  5130.2   547.8  5242.4  552.26  5372.4  554.68  5457.4  555.24    5717  558.02
#Mann= 8 ,-1 , 0
  3691.5    .035       0  4014.4     .07       0  4699.6      .1       0
  5006.1     .05       0  5014.9      .1       0  5097.3     .07       0
  5130.2     .12       0  5457.4     .07       0
Bank Sta=5006.1,5014.9
XS Rating Curve= 0 ,0
Exp/Cntr=0.3,0.1

Type RM Length L Ch R = 1 ,81940   ,503,503,503
BEGIN DESCRIPTION:
B19432
END DESCRIPTION:
XS GIS Cut Line= 3
      2328929.86     13785276.13      2327608.85     13785549.44
      2327146.85     13785913.84
#Sta/Elev= 30
    3872  552.84  3941.9  554.23  4017.9  553.85  4042.3  553.41  4111.8  549.66
    4238  546.49  4367.1  542.05  4448.8  542.49  4489.7  541.64  4534.2  542.14
  4876.5   540.3  4898.1  539.98    4939  537.41  4969.6  537.55  4975.8  533.76
    4981  534.24  4985.6  529.18  4986.1  528.68  4994.5  529.18  5000.3  529.67
  5010.5  535.42  5020.7  536.76  5026.1  538.57  5031.2  538.77  5051.3  544.01
  5112.6  547.12  5151.5   547.4    5256  548.59  5413.1   553.1  5809.4  557.03
#Mann= 6 ,-1 , 0
    3872    .035       0  4017.9     .07       0  4876.5     .12       0
  4985.6     .05       0  4994.5     .12       0  5151.5     .07       0
Bank Sta=4985.6,4994.5
XS Rating Curve= 0 ,0
Exp/Cntr=0.3,0.1

Type RM Length L Ch R = 1 ,81437   ,465,465,465
BEGIN DESCRIPTION:
B19431
END DESCRIPTION:
XS GIS Cut Line= 3
      2328897.29     13785022.35      2327595.84     13785159.01
      2327166.37     13785653.55
#Sta/Elev= 30
    4064  552.29  4146.7  554.61  4208.5   553.6  4247.3  552.71  4408.2  544.83
  4428.9  545.02  4629.4  539.45  4760.1  539.34  4806.4  538.17  4880.8  539.11
  4981.3  538.19  4991.4   537.5  4997.7  533.47  5002.8  534.08  5006.9  530.41
  5007.4  529.91    5016  530.41  5031.6  531.57  5051.7  535.84  5081.9  537.07
  5142.2  537.06  5182.4  534.65  5202.5  536.35  5238.3   537.3  5303.1  539.96
  5333.2  539.98  5384.3  544.36  5433.7  546.73  5682.5  551.83  6027.6  555.16
#Mann= 5 ,-1 , 0
    4064    .035       0  4208.5     .07       0  5006.9     .05       0
    5016     .07       0  5238.3     .07       0
Bank Sta=5006.9,5016
XS Rating Curve= 0 ,0
Exp/Cntr=0.3,0.1

Type RM Length L Ch R = 1 ,80972   ,483,483,483
BEGIN DESCRIPTION:
B19430
END DESCRIPTION:
XS GIS Cut Line= 2
      2328897.25      13784788.1      2327069.42     13784710.04
#Sta/Elev= 30
  3840.2  549.84  4012.6  549.23  4062.7  546.32  4082.7  543.33  4102.7  542.82
  4122.7  545.47  4152.7   543.5  4301.3  540.38    4433  537.28  4691.8   534.9
  4775.4  534.54  4846.9  534.29  4883.4  532.88  4913.4  533.02  4943.5  534.75
    4963  532.01    4968  532.87  4978.7  527.61  4979.2  527.11  4988.3  527.61
  5008.6  530.63  5013.5  531.96  5023.5  537.33  5043.5  540.29  5083.6  540.64
  5183.7  544.53  5295.5  545.69  5479.9  548.68    5524  549.33  5669.7  550.21
#Mann= 11 ,-1 , 0
  3840.2    .035       0  4301.3     .07       0  4691.8     .12       0
  4775.4     .07       0  4846.9     .12       0  4978.7     .05       0
  4988.3     .12       0  5008.6     .07       0  5295.5     .05       0
  5479.9     .07       0    5524     .05       0
Bank Sta=4978.7,4988.3
XS Rating Curve= 0 ,0
Exp/Cntr=0.3,0.1

Type RM Length L Ch R = 1 ,80489   ,490,490,490
BEGIN DESCRIPTION:
B19429
END DESCRIPTION:
XS GIS Cut Line= 3
       2328858.2       13784710.        2327739.      13784423.7
      2326860.51     13784508.29
#Sta/Elev= 30
  4140.5  548.65    4184  548.44  4345.4  545.15    4567  536.33  4583.4  537.97
  4588.6  536.29    4598   537.7  4787.5   534.4  4931.5  534.71  4954.1  534.94
  4969.6  535.15  4979.9   531.7  4986.5  523.98  4990.6  526.67  4991.6  527.32
  4995.7  521.45  4996.2  520.95  5005.3  521.45  5027.3  526.85  5032.4  523.95
  5051.7  531.06  5173.5  532.61  5237.9  532.21  5295.2  537.25  5353.5   538.8
  5681.1   546.4  5711.7  547.72  5827.6  547.42  6173.9  548.22  6178.3  548.21
#Mann= 14 ,-1 , 0
  4140.5    .035       0    4184     .07       0  4345.4    .035       0
  4931.5     .07       0  4954.1     .12       0  4990.6     .07       0
  4995.7     .05       0  5005.3     .07       0  5051.7     .12       0
  5173.5     .07       0  5353.5     .05       0  5681.1    .035       0
  5827.6     .05       0  6173.9     .07       0
Bank Sta=4995.7,5005.3
XS Rating Curve= 0 ,0
Exp/Cntr=0.3,0.1

Type RM Length L Ch R = 1 ,79999   ,685,685,685
BEGIN DESCRIPTION:
B19428
END DESCRIPTION:
XS GIS Cut Line= 4
      2329027.43     13784404.18      2328292.11     13784013.74
       2327647.9     13784117.86      2326984.12     13784339.12
#Sta/Elev= 30
  3643.1  542.11  3863.8  539.61    4190  536.56  4288.6  537.21  4354.6  534.89
  4402.7  535.01    4493  533.56  4538.2  529.88  4551.5  529.65  4655.1  529.89
  4695.6  528.56  4817.1  530.32  4858.3  529.18  4918.4  529.62  4958.9  528.49
  4984.5  522.23    4985  521.73  4994.2  522.23  4999.5  523.58  5009.6  530.04
  5015.5  531.09    5040  532.65  5151.5  534.58  5247.2  538.97  5325.5   540.3
  5415.1  545.31  5533.7  546.41  5673.9  546.23  5731.3  547.23  5827.9  546.57
#Mann= 11 ,-1 , 0
  3643.1     .07       0  3863.8     .12       0  4402.7    .035       0
  4538.2     .07       0  4551.5    .035       0  4858.3     .07       0
  4984.5     .05       0  4994.2     .07       0  5151.5     .05       0
  5533.7    .035       0  5673.9     .05       0
Bank Sta=4984.5,4994.2
XS Rating Curve= 0 ,0
Exp/Cntr=0.3,0.1

Type RM Length L Ch R = 1 ,79314   ,531,531,531
BEGIN DESCRIPTION:
B19427
END DESCRIPTION:
XS GIS Cut Line= 3
      2328806.16      13783519.2      2327843.11     13783753.46
      2327094.82     13784124.35
#Sta/Elev= 30
  4345.5  538.81  4709.1  534.44  4921.6   533.8  4953.9  532.32  4964.2  530.64
  4973.1  525.46  4981.8  519.95  4982.3  519.45  4991.6  519.95  4995.1  523.96
  5005.4  525.97  5028.5   525.8  5046.5  527.18  5136.7  527.43  5195.4  527.53
  5262.6  526.07    5310  528.04  5395.1  530.17    5441  530.79  5508.3  528.41
  5574.6     529  5635.9  530.19  5715.6  536.29  5754.9  537.68  5782.9  540.44
  5859.1  544.07  5962.2  546.74  6064.9  545.16    6127  544.15  6171.8  545.67
#Mann= 11 ,-1 , 0
  4345.5     .05       0  4709.1    .035       0  4921.6     .07       0
  4973.1     .12       0  4981.8     .05       0  4991.6     .12       0
  5136.7     .07       0    5310     .05       0  5395.1     .07       0
  5574.6     .05       0  6064.9    .035       0
Bank Sta=4981.8,4991.6
XS Rating Curve= 0 ,0
Exp/Cntr=0.3,0.1

Type RM Length L Ch R = 1 ,78783   ,583,583,583
BEGIN DESCRIPTION:
B19426
END DESCRIPTION:
XS GIS Cut Line= 3
      2328604.43      13783057.2      2327699.95     13783493.17
      2327244.46      13783987.7
#Sta/Elev= 30
  4134.2  541.91  4160.6  540.91  4167.9  540.64  4377.8   534.2  4516.7  532.22
    4651  529.13  4665.6  526.37  4688.2  525.17  4827.5  523.93  4993.3  522.96
  5005.5  518.51    5006  518.01  5015.3  518.51  5038.6  523.42  5128.1  523.73
  5142.9  522.06  5150.3  523.17    5157  527.27  5178.6  528.39  5319.8  531.46
  5341.4  530.19  5355.5  528.35  5362.3  525.67  5376.5  525.03  5404.9  527.86
  5461.6  527.98  5496.7  531.85    5564  536.04  5681.1  544.28  5810.6  544.87
#Mann= 10 ,-1 , 0
  4134.2     .05       0  4160.6     .07       0  4167.9     .05       0
  4516.7     .07       0    4651    .035       0  4827.5     .12       0
  5005.5     .05       0  5015.3     .12       0  5128.1     .07       0
    5564     .05       0
Bank Sta=5005.5,5015.3
XS Rating Curve= 0 ,0
Exp/Cntr=0.3,0.1

Type RM Length L Ch R = 1 ,78200   ,513,513,513
BEGIN DESCRIPTION:
Mill Creek 96.0
END DESCRIPTION:
XS GIS Cut Line= 3
      2328024.96     13782925.02        2327775.       13783025.
      2327275.01     13783824.99
#Sta/Elev= 30
  4726.4  528.73  4774.1  528.43  4866.4     525  4873.1  524.49  4878.5  521.75
  4899.6  520.95    4927  522.07  4951.2  520.53  4974.1   515.9  4975.9  513.58
  4976.4  513.08  4985.7  513.58  4998.6  514.13  5009.2   520.2  5018.6  521.24
  5098.4  522.18    5099  522.12  5148.9  521.69  5286.3  526.74  5495.6  527.48
  5511.5  529.35  5517.4  527.86  5526.3  528.41  5538.7  524.92  5584.6  524.59
  5611.8  528.08  5663.7  528.18  5782.5  534.76  5873.6  541.23    5939  543.25
#Mann= 9 ,-1 , 0
  4726.4     .05       0  4774.1     .07       0  4899.6    .035       0
  4975.9    .035       0  4985.7    .035       0  5098.4     .07       0
    5099     .05       0  5495.6     .07       0  5782.5     .05       0
Bank Sta=4975.9,4985.7
XS Rating Curve= 0 ,0
Exp/Cntr=0.3,0.1

Type RM Length L Ch R = 1 ,77687   ,405,405,405
BEGIN DESCRIPTION:
B19425
END DESCRIPTION:
XS GIS Cut Line= 3
      2328487.34      13782530.1      2327550.29     13782842.45
      2326964.63     13783584.29
#Sta/Elev= 30
  3723.7  540.82  3780.4  538.49    3791  538.28  3901.7  534.16  4083.4  529.49
  4438.8  527.47  4481.1  527.72  4639.2  523.92  4745.4  522.76    4795  519.74
  4806.5  519.93  4844.7  518.02  4880.3  519.49  4944.1   519.8  4987.4  516.45
    4995  515.42  4996.9  513.48  4997.4  512.98  5006.8  513.48  5016.3  521.95
  5041.1  523.53    5066  524.24  5150.9  522.55  5250.3  525.93  5293.6  524.85
  5357.8  527.58  5442.7  535.63  5599.8  541.28  5651.5  542.21  5656.6  542.29
#Mann= 12 ,-1 , 0
  3723.7     .05       0  3780.4     .07       0    3791     .05       0
  3901.7     .07       0  4083.4     .05       0  4438.8     .07       0
  4639.2    .035       0  4806.5     .12       0  4996.9     .05       0
  5006.8     .12       0  5041.1     .05       0  5651.5    .035       0
Bank Sta=4996.9,5006.8
XS Rating Curve= 0 ,0
Exp/Cntr=0.3,0.1

Type RM Length L Ch R = 1 ,77282   ,477,477,477
BEGIN DESCRIPTION:
B19424
END DESCRIPTION:
XS GIS Cut Line= 3
      2328448.27      13782432.5       2327016.7      13782796.9
      2326079.86     13783232.79
#Sta/Elev= 30
  3789.4  537.67  4008.4  531.32  4109.5  529.06    4160   528.3  4464.6  526.56
  4805.7  521.94  4845.3  522.09  4935.2  516.75  4979.4  517.21  4995.2  512.55
  5005.4  512.13  5005.9  511.63  5015.5  512.13  5041.4  516.14  5134.2  520.82
  5270.3  522.06  5296.9  522.92  5302.4     525  5319.8  523.34  5325.3  525.75
  5348.2  524.28  5416.8   530.1  5446.1  534.86  5478.1  538.85  5586.6  539.94
  5764.8  538.44  5807.7  540.17  6011.4  543.53  6231.7  552.18  6299.9  555.48
#Mann= 14 ,-1 , 0
  3789.4     .07       0  4008.4     .05       0  4109.5     .07       0
    4160     .05       0  4464.6     .07       0  4805.7    .035       0
  4935.2     .12       0  5005.4     .05       0  5015.5     .12       0
  5446.1    .035       0  5586.6     .07       0  5807.7     .05       0
  6011.4     .12       0  6231.7     .07       0
Bank Sta=5005.4,5015.5
XS Rating Curve= 0 ,0
Exp/Cntr=0.3,0.1
