HEC-RAS study Mill Creek.prj: Mill Creek Base Level Engineering

--- Mill Creek.g01 (geometry) --- (continued)

Type RM Length L Ch R = 1 ,76805   ,636,636,636
BEGIN DESCRIPTION:
B19423
END DESCRIPTION:
XS GIS Cut Line= 3
      2328435.23     13782367.43      2326886.56     13782510.59
      2326139.12     13782777.06
#Sta/Elev= 30
    3466  536.36  3837.8  526.79  4019.6  525.98  4126.4  524.38  4219.4  521.42
  4390.2  522.88    4676  519.74  4731.6  518.82  4781.8  513.05  4811.9   514.8
  4852.1  515.14  4872.2  513.72  4910.6  514.88  4962.6  515.42  5006.3  512.18
  5006.8  511.68  5016.4  512.18  5019.5  515.39  5024.8  515.39  5033.5  520.25
  5136.5  520.77  5179.1  522.39  5192.8  522.88  5235.3  530.95  5267.1  534.24
  5352.8  534.75  5458.2  534.41    5501  536.69  5521.2  535.09  5814.8  543.74
#Mann= 9 ,-1 , 0
    3466     .07       0  4019.6     .05       0  4126.4     .07       0
    4676    .035       0  4910.6     .12       0  5006.3     .05       0
  5016.4     .12       0  5179.1    .035       0  5352.8     .07       0
Bank Sta=5006.3,5016.4
XS Rating Curve= 0 ,0
Exp/Cntr=0.3,0.1

Type RM Length L Ch R = 1 ,76169   ,341,341,341
BEGIN DESCRIPTION:
B19422
END DESCRIPTION:
XS GIS Cut Line= 3
      2328422.22     13782042.07      2326867.04     13782204.75
      2326230.42     13782380.14
#Sta/Elev= 30
  3593.8  531.25  3741.8  526.89  3892.6  525.04  4214.4  524.06  4485.9  519.27
  4636.7  520.23  4852.6  517.97  4978.5  517.35  4998.6   508.5  5009.7  506.28
  5010.2  505.78  5019.8  506.28    5069  512.75  5089.1  521.73  5131.7  528.13
    5156  530.68  5242.6  530.77  5250.1  530.55  5255.3  528.16  5289.7  527.16
  5294.9  524.74  5324.1  527.02  5329.3  525.28  5363.7  529.85    5398  531.45
  5482.8     533  5625.1  529.99  5738.6  531.84  5750.8  533.76  5817.8   532.5
#Mann= 6 ,-1 , 0
  3593.8     .07       0  4852.6     .12       0  5009.7     .05       0
  5019.8     .12       0  5131.7    .035       0  5482.8     .07       0
Bank Sta=5009.7,5019.8
XS Rating Curve= 0 ,0
Exp/Cntr=0.3,0.1

Type RM Length L Ch R = 1 ,75828   ,523,523,523
BEGIN DESCRIPTION:
B19421
END DESCRIPTION:
XS GIS Cut Line= 2
      2328155.48     13781547.52      2326379.47     13782022.42
#Sta/Elev= 30
  3777.6   528.5  3980.4  521.25  4161.1  520.91  4264.6  515.96  4330.5  515.89
  4357.8  514.15  4378.5  514.98  4405.5  511.36  4440.4  510.66  4492.3  513.46
  4565.7   514.1  4585.5     513    4658  515.81  4675.5   514.4  4694.7  516.04
  4709.7  517.51  4750.5  514.53  4937.4  514.65  4950.8  513.91  4985.8  503.16
  4986.3  502.66  4995.9  503.16  4999.6  503.87  5009.9  511.47  5025.7  518.23
  5085.3  521.85  5206.6  526.82  5387.4  531.04  5519.6  531.63    5616  531.21
#Mann= 7 ,-1 , 0
  3777.6     .07       0  4694.7     .12       0  4985.8     .05       0
  4995.9     .12       0  5085.3     .07       0  5387.4    .035       0
  5519.6     .07       0
Bank Sta=4985.8,4995.9
XS Rating Curve= 0 ,0
Exp/Cntr=0.3,0.1

Type RM Length L Ch R = 1 ,75305   ,529,529,529
BEGIN DESCRIPTION:
B19420
END DESCRIPTION:
XS GIS Cut Line= 3
      2328148.96     13781371.83      2327413.64      13781254.7
      2326328.46     13781761.55
#Sta/Elev= 30
    3911  528.03  4026.4  522.57  4289.7   517.7  4380.8  514.06  4573.2  513.01
  4766.3  514.58    4871  513.48  4896.9  514.15  4926.3  513.33  4931.8  511.94
  4949.1  510.98  4954.6  509.35  4977.5  508.59  4985.2  505.77  4989.7  505.21
  4990.2  504.71    5000  505.21  5000.4  505.97  5029.3  509.78  5062.5  509.69
  5074.4  508.38    5091  509.89  5097.3  510.77  5188.7  509.95  5250.1     513
  5382.5  523.45  5481.9  527.99  5713.6     530  5816.1  529.17  5853.3   529.1
#Mann= 6 ,-1 , 0
    3911     .07       0    4871     .12       0  4989.7     .05       0
    5000     .12       0    5091     .07       0  5816.1    .035       0
Bank Sta=4989.7,5000
XS Rating Curve= 0 ,0
Exp/Cntr=0.3,0.1

Type RM Length L Ch R = 1 ,74776   ,339,339,339
BEGIN DESCRIPTION:
B19419
END DESCRIPTION:
XS GIS Cut Line= 4
      2328122.91     13781280.72        2327290.     13780903.31
      2326691.34     13781150.59      2326288.97     13781488.06
#Sta/Elev= 30
  3628.1  525.66  3774.6  520.78  3964.9  517.96  4097.9  512.98  4218.7  511.28
  4310.1  510.51  4542.5  511.87    4586  513.54  4591.4  512.31  4615.3  512.95
  4764.3  510.17  4863.2  511.95    4924  511.34  4959.1     506  4977.2  504.59
  4982.6  505.53  4991.5   501.1  5001.1  498.32  5001.4  497.29  5001.9  496.79
  5011.7  497.29  5030.5  507.93  5067.3  508.94  5107.6  507.85  5166.3  512.62
  5254.4  514.71  5297.3  519.86  5325.9  521.84  5453.4  525.03  5715.4  525.98
#Mann= 4 ,-1 , 0
  3628.1     .07       0  4863.2      .1       0  5001.4     .05       0
  5011.7    .035       0
Bank Sta=5001.4,5011.7
XS Rating Curve= 0 ,0
Exp/Cntr=0.3,0.1

Type RM Length L Ch R = 1 ,74437   ,613,613,613
BEGIN DESCRIPTION:
B19418
END DESCRIPTION:
XS GIS Cut Line= 4
      2327999.26     13781124.55      2326912.59     13780688.58
      2326489.62     13780942.36      2326222.81     13781378.37
#Sta/Elev= 30
  3483.6  520.05  3671.4  517.14  3841.7  511.51  4016.2  510.25  4307.1  511.74
  4523.4  507.88  4576.4  502.38  4608.8  503.53  4630.3  505.83  4663.5  504.47
  4694.3  506.28  4724.3  504.68  4758.4   503.8  4791.4  504.95  4896.6  507.06
  4964.5  505.82  5001.4  504.14  5017.6  500.38  5018.1  499.88  5027.9  500.38
  5028.6  504.34  5036.5  507.11  5123.8  505.61  5145.2  511.49  5147.5  514.39
  5152.2  514.39  5167.3  518.89  5234.3  520.14  5583.2  523.97  5658.9  523.58
#Mann= 8 ,-1 , 0
  3483.6     .07       0  4523.4    .035       0  4663.5      .1       0
  4724.3    .035       0  4791.4     .07       0  5017.6     .05       0
  5027.9     .07       0  5234.3     .05       0
Bank Sta=5017.6,5027.9
XS Rating Curve= 0 ,0
Exp/Cntr=0.3,0.1

Type RM Length L Ch R = 1 ,73824   ,599,599,599
BEGIN DESCRIPTION:
B19417
END DESCRIPTION:
XS GIS Cut Line= 4
      2327927.68     13781033.44      2326945.12     13780486.85
      2326255.36     13780584.46      2326183.92     13781331.36
#Sta/Elev= 30
  3654.2  518.19  3771.7   516.8  3862.3  512.29  3933.2  510.59    4139  509.48
  4355.1  510.72  4572.7  505.49  4635.2  505.47  4691.3  506.66  4756.5     503
  4781.1  503.59  4788.8  505.97  4813.3  507.69  4859.5  508.57  4932.5  504.79
  4980.7  505.31  5000.9   499.4  5010.4   498.4  5010.9   497.9  5020.7   498.4
  5031.2  502.92  5202.9  506.39  5228.1  508.63  5233.7  512.15  5263.5   514.3
  5312.7  513.06  5412.5   512.9  5499.3     513    5978  517.48  6225.5  522.23
#Mann= 9 ,-1 , 0
  3654.2     .07       0  4635.2    .035       0  4813.3     .07       0
  4932.5      .1       0  5010.4     .05       0  5020.7      .1       0
  5312.7     .05       0  5412.5     .07       0  5499.3     .05       0
Bank Sta=5010.4,5020.7
XS Rating Curve= 0 ,0
Exp/Cntr=0.3,0.1

Type RM Length L Ch R = 1 ,73225   ,1546,1546,1546
BEGIN DESCRIPTION:
Mill Creek 90.0
END DESCRIPTION:
XS GIS Cut Line= 3
       2327908.2     13780961.89      2326548.18     13780246.09
      2325098.55     13780564.62
#Sta/Elev= 30
  3183.1  517.26  3272.3  516.22  3435.3  510.16  3850.3  510.32  4122.5  505.26
  4181.2  506.63    4249  503.09  4279.7  506.13  4308.5  506.19  4465.5  505.35
    4621  505.64    4701  501.96  4836.2  504.39  4948.5  501.67  4972.6  497.03
    4974  494.51  4974.5  494.01  4984.4  494.51  4997.4  505.55  5009.9  508.23
  5425.5  508.61  5584.6  505.84  5626.4  498.53  5644.7  504.45  5670.2  504.38
    5712   508.4  5944.7  524.14    6111  531.59  6148.8  534.05  6204.2  536.68
#Mann= 13 ,-1 , 0
  3183.1     .07       0  4122.5    .035       0  4308.5     .07       0
  4465.5      .1       0    4974     .05       0  4984.4      .1       0
  4997.4     .05       0  5425.5     .07       0  5584.6     .12       0
    5712     .07       0  5944.7     .12       0    6111     .07       0
  6148.8     .12       0
Bank Sta=4974,4984.4
XS Rating Curve= 0 ,0
Exp/Cntr=0.3,0.1

Type RM Length L Ch R = 1 ,71679   ,716,716,716
BEGIN DESCRIPTION:
Mill Creek 89.0
END DESCRIPTION:
XS GIS Cut Line= 3
      2327875.63     13780896.78      2327003.69     13779790.59
      2325136.17     13780304.64
#Sta/Elev= 30
  3457.5  516.43  3836.8  508.06  4383.2  507.57  4595.8  507.29  4641.8  507.21
    4866  504.37  4901.2  495.73  4982.1  496.43  5014.8  496.53    5015  491.75
  5015.5  491.25  5025.4  491.75  5049.2  500.52  5281.5  509.95  5341.8  507.01
  5362.5  502.19  5388.4  505.45  5395.1  502.56  5424.3  506.92  5517.6  505.75
  5879.4  504.19  6018.6  502.57  6078.2  502.76  6098.9   496.5  6110.9   497.1
  6119.7  500.98  6179.7  504.96  6260.4  506.09  6554.8  517.61    6803  534.48
#Mann= 11 ,-1 , 0
  3457.5     .07       0  4383.2    .035       0  4595.8     .07       0
  4641.8    .035       0  4982.1      .1       0    5015     .05       0
  5025.4      .1       0  5517.6     .05       0  5879.4     .07       0
  6018.6     .12       0  6260.4     .07       0
Bank Sta=5015,5025.4
XS Rating Curve= 0 ,0
Exp/Cntr=0.3,0.1

Type RM Length L Ch R = 1 ,70963   ,732,732,732
BEGIN DESCRIPTION:
Mill Creek 88.0
END DESCRIPTION:
XS GIS Cut Line= 3
      2327817.08     13778677.86      2326125.22     13779653.93
      2325201.22     13779927.23
#Sta/Elev= 30
  3912.4   529.3  4020.2  528.46  4132.6  523.56  4191.5  528.23  4216.4  521.52
  4240.3  512.38  4589.4  501.78  4682.9  498.52  4798.6   496.9  4893.8  497.02
  4915.3  489.63  4936.9  495.57    4980  495.96  4990.5  489.33    4991  488.83
    5001  489.33  5054.6   500.1  5094.2  501.61  5300.2  501.25  5521.5   501.8
  5663.3  500.48  5785.5  502.03  6001.4  499.67  6027.8   493.3  6132.8  503.07
  6337.2  505.59  6362.6  505.98  6389.7  506.19  6795.6   519.4  6829.2  520.95
#Mann= 17 ,-1 , 0
  3912.4     .05       0  4020.2     .12       0  4216.4     .07       0
  4589.4     .12       0  4682.9     .07       0  4798.6      .1       0
  4990.5     .05       0    5001      .1       0  5094.2     .07       0
  5300.2    .035       0  5521.5     .07       0  5663.3     .05       0
  5785.5     .12       0  6337.2     .07       0  6362.6     .12       0
  6389.7     .07       0  6795.6     .12       0
Bank Sta=4990.5,5001
XS Rating Curve= 0 ,0
Exp/Cntr=0.3,0.1

Type RM Length L Ch R = 1 ,70231   ,563,563,563
BEGIN DESCRIPTION:
Mill Creek 87.0
END DESCRIPTION:
XS GIS Cut Line= 3
      2326743.41     13778411.03       2326385.5     13779230.97
      2325299.39     13779848.82
#Sta/Elev= 30
  4603.7  523.65  4665.1  517.82  4683.1  519.07  4695.3  516.85  4783.2  514.99
  4865.8  513.41    4939  513.72  4962.4  511.13  4971.9   505.6  5001.2  487.75
  5001.7  487.25  5017.2  487.75  5032.6  494.75  5047.2     495  5077.9  493.58
  5113.8   493.9  5137.2  491.54    5184  495.62  5363.4  498.61  5647.1  499.34
  5694.3  499.57  5736.9  497.33    5752  499.08  5780.2  491.38  5801.8  496.89
  5877.5  498.47  6264.5  506.69  6380.3  507.18  6640.7  511.16  6747.9  515.49
#Mann= 14 ,-1 , 0
  4603.7     .07       0  4783.2     .05       0  4865.8     .12       0
  4971.9      .1       0  5001.2     .05       0  5017.2      .1       0
  5047.2     .12       0  5077.9     .07       0  5363.4    .035       0
  5647.1     .07       0  5694.3     .12       0  5877.5     .07       0
  6380.3     .12       0  6640.7     .07       0
Bank Sta=5001.2,5017.2
XS Rating Curve= 0 ,0
Exp/Cntr=0.3,0.1

Type RM Length L Ch R = 1 ,69668   ,489,489,489
BEGIN DESCRIPTION:
Mill Creek 86.0
END DESCRIPTION:
XS GIS Cut Line= 3
      2326665.34     13778313.43      2325995.07     13779107.33
      2325272.74     13779797.13
#Sta/Elev= 30
  4181.8  524.45    4254   524.1  4296.8  517.25  4362.9   515.3  4381.4  515.68
  4403.4  519.97    4432  517.06  4614.3  512.93  4633.9  511.95    4740  506.65
  4914.4  492.76  4950.2  492.89  4984.7     492  5005.2  488.13  5005.7  487.63
  5021.3  488.13  5041.9  493.73  5062.7  492.31  5084.8   497.2  5108.4   496.1
    5245   498.1  5261.3  498.46  5325.3  495.18  5383.2  495.22  5396.1  490.95
  5431.3   498.7  5714.4  501.98  5960.3  508.82  6212.8  515.94  6219.6  516.06
#Mann= 14 ,-1 , 0
  4181.8     .07       0  4362.9     .05       0  4614.3      .1       0
  4633.9     .05       0    4740      .1       0  4950.2    .035       0
  5005.2    .035       0  5021.3    .035       0  5108.4     .07       0
    5245     .12       0  5261.3      .1       0  5383.2     .07       0
  5960.3     .12       0  6212.8     .07       0
Bank Sta=5005.2,5021.3
XS Rating Curve= 0 ,0
Exp/Cntr=0.3,0.1

Type RM Length L Ch R = 1 ,69179   ,662,662,662
BEGIN DESCRIPTION:
Mill Creek 84.0
END DESCRIPTION:
XS GIS Cut Line= 3
      2326502.66     13778163.77      2325643.69       13778808.
      2325071.01      13779146.4
#Sta/Elev= 30
  4008.2  525.91  4056.7  524.74  4065.1  522.23  4071.3  524.51  4079.6  522.13
  4085.9  523.89  4120.7  521.06  4200.5  519.78  4256.7  513.29  4280.3  514.66
  4310.1  512.23  4406.2  508.09  4532.1  503.13  4865.1  494.85  4921.3  490.09
  4941.6  491.61  4985.9  493.22  4992.8  491.67  4998.7  486.86  4999.2  486.36
  5014.8  486.86  5021.3  490.33  5035.9  491.73  5102.4  492.98  5128.9  492.75
  5142.8  487.77    5166  493.23  5286.7  495.48  5616.8  522.14  5747.1  526.55
#Mann= 13 ,-1 , 0
  4008.2    .035       0  4120.7     .07       0  4280.3    .035       0
  4310.1     .05       0  4406.2    .035       0  4532.1     .05       0
  4941.6    .035       0  4998.7    .035       0  5014.8    .035       0
  5102.4      .1       0  5142.8     .07       0  5286.7     .05       0
  5616.8     .07       0
Bank Sta=4998.7,5014.8
XS Rating Curve= 0 ,0
Exp/Cntr=0.3,0.1

Type RM Length L Ch R = 1 ,68517   ,454,454,454
BEGIN DESCRIPTION:
Mill Creek 83.0
END DESCRIPTION:
XS GIS Cut Line= 3
      2326339.99     13778085.69        2325175.       13778475.
      2324974.97     13778525.01
#Sta/Elev= 30
    3767  523.22  3860.1  518.46  3942.3  515.52  4025.3  509.16  4063.4  504.43
  4088.6     505    4095  505.83  4100.2  508.78  4126.6  509.47  4131.8   511.5
  4151.8  511.36  4189.7  504.28    4195  499.13  4221.3  495.27  4320.8  495.13
  4689.6  494.25  4805.5  489.07  4837.2  491.17  4902.3  491.54    4996  491.38
  5005.6  489.98  5009.6   483.5  5010.1     483  5027.5   483.5  5046.9  494.72
  5059.7  499.95  5088.1  507.51  5108.7  515.14  5142.2  518.99  5201.5  521.53
#Mann= 7 ,-1 , 0
    3767    .035       0  3860.1     .07       0  4320.8     .05       0
  4902.3     .07       0    4996     .05       0  5009.6     .05       0
  5027.5     .05       0
Bank Sta=5009.6,5027.5
XS Rating Curve= 0 ,0
Exp/Cntr=0.3,0.1

Type RM Length L Ch R = 1 ,68063   ,434,434,434
BEGIN DESCRIPTION:
Mill Creek 82.0
END DESCRIPTION:
XS GIS Cut Line= 3
      2326235.81     13778040.16        2325025.       13778075.
      2324491.88     13778209.35
#Sta/Elev= 30
    3789  519.24  3806.8  518.43  3909.9  513.16  4009.9   505.4  4239.8  498.82
    4320  497.43  4421.6  506.91  4440.1  507.23    4477  504.53    4482  501.22
  4510.1  493.27  4550.1   488.9  4590.1  488.93  4610.1  493.63  4618.8  493.59
  4895.2  488.57  4920.3  487.81  4980.3  490.65  4990.3  489.09  4997.8  484.13
  5014.4  481.45  5014.9  480.95  5032.4  481.45  5041.6  492.61  5059.4  496.14
  5064.5  498.63    5092  501.26  5124.1  506.51  5352.1  514.73  5550.1  515.57
#Mann= 9 ,-1 , 0
    3789    .035       0  3806.8     .07       0  4239.8     .12       0
  4421.6     .07       0  4618.8     .05       0  4895.2     .07       0
  5014.4     .05       0  5032.4     .07       0    5092     .05       0
Bank Sta=5014.4,5032.4
XS Rating Curve= 0 ,0
Exp/Cntr=0.3,0.1

Type RM Length L Ch R = 1 ,67629   ,515,515,515
BEGIN DESCRIPTION:
Mill Creek 81.0
END DESCRIPTION:
XS GIS Cut Line= 3
      2326313.89     13777487.05       2324927.9     13777662.74
      2324625.01       13777825.
#Sta/Elev= 30
  3650.2  531.73  3871.9     519  3931.3  515.43  4052.3   519.5  4203.5  510.02
  4284.1  501.43    4395  495.61  4750.6  487.84  4750.7  487.84  4850.2  488.41
    4899  486.98  4949.9  489.19  4979.6  488.08  4990.8  480.73  4991.3  480.23
  5008.9  480.73  5009.9  486.62  5025.3  492.49  5030.3  491.78  5049.8  497.43
  5118.6  497.76  5125.3  496.98  5130.9   493.3  5152.7  492.66  5163.3  493.59
  5191.1  502.39  5229.2  505.25  5294.3   489.9  5322.8  501.42  5390.9  503.31
#Mann= 12 ,-1 , 0
  3650.2     .12       0  3871.9     .07       0  4750.6      .1       0
  4750.7     .12       0  4850.2      .1       0  4949.9     .12       0
  4990.8     .05       0  5008.9     .12       0  5049.8     .07       0
  5152.7     .12       0  5163.3     .07       0  5294.3     .05       0
Bank Sta=4990.8,5008.9
XS Rating Curve= 0 ,0
Exp/Cntr=0.3,0.1

Type RM Length L Ch R = 1 ,67114   ,691,691,691
BEGIN DESCRIPTION:
Mill Creek 80.0
END DESCRIPTION:
XS GIS Cut Line= 3
      2325575.03     13776974.97        2325225.       13777325.
      2324225.04     13777624.99
#Sta/Elev= 30
  4501.3  522.27    4557   518.7  4642.8  508.11    4671  502.75  4741.8  495.88
  4826.6  494.41  4925.6  489.22  4953.9   489.7  4982.2  483.37  4983.7  479.96
  4984.2  479.46  5001.9  479.96  5006.8  481.47  5012.8  486.58  5027.6  487.46
    5059  486.32  5155.5  488.99  5287.8   488.6  5326.5  491.33  5560.1  494.12
  5716.7  498.52  5776.7  499.17  5795.1  497.27    5842  497.85  5886.3  507.14
  5904.6  508.37  5952.5   504.3  5967.3  500.15  6031.7  504.19  6040.3  504.24
#Mann= 7 ,-1 , 0
  4501.3     .12       0    4557      .1       0  4983.7     .05       0
  5001.9      .1       0  5326.5     .07       0  5795.1     .12       0
  6031.7     .07       0
Bank Sta=4983.7,5001.9
XS Rating Curve= 0 ,0
Exp/Cntr=0.3,0.1

Type RM Length L Ch R = 1 ,66423   ,672,672,672
BEGIN DESCRIPTION:
B19416
END DESCRIPTION:
XS GIS Cut Line= 3
      2325787.02     13776547.08      2324565.94     13777082.95
      2323854.34     13777574.92
#Sta/Elev= 30
  4275.8  532.57  4306.6  527.53  4438.9  523.03  4486.6  519.88  4533.9  521.28
  4562.1   528.2  4594.7  522.74  4647.7  520.62  4731.1  519.87  4763.5  511.88
  4845.8  502.81  4905.6  496.92  4928.9  490.65  4998.8  482.56  5000.8  478.98
  5001.3  478.48    5019  478.98  5033.3  484.33  5083.1  485.56  5192.4  487.38
  5222.6  487.76  5550.8   490.2  5797.2   493.6  6072.4  497.09  6208.7  501.75
  6230.4  502.69  6252.5  507.66  6272.7  510.72  6308.5  506.71  6474.4  512.48
#Mann= 15 ,-1 , 0
  4275.8     .05       0  4438.9     .07       0  4533.9     .05       0
  4647.7     .07       0  4763.5     .12       0  4845.8      .1       0
  5000.8     .05       0    5019      .1       0  5083.1     .07       0
  5192.4     .12       0  5222.6     .07       0  5550.8     .12       0
  5797.2     .07       0  6208.7     .12       0  6252.5     .07       0
Bank Sta=5000.8,5019
XS Rating Curve= 0 ,0
Exp/Cntr=0.3,0.1

Type RM Length L Ch R = 1 ,65751   ,587,587,587
BEGIN DESCRIPTION:
B19415
END DESCRIPTION:
XS GIS Cut Line= 3
      2325778.23     13776011.21      2324135.49     13776793.05
      2323081.34     13777407.97
#Sta/Elev= 30
  3711.7  532.29    4169  511.18    4271  509.87  4401.7  500.44  4429.9  507.54
  4475.3  501.27  4725.4  488.21  4798.8  484.84  4912.4  484.55  4963.3  485.39
  4976.9  476.41  4977.4  475.91  4995.1  476.41    5000  481.53  5008.7   483.7
  5057.2  486.41  5128.2  487.83  5425.3  490.71  5614.2  497.12  5867.7  510.41
  5953.5   511.7  6167.4  512.93  6294.4  514.72  6401.9  512.19  6440.4  515.81
  6500.7  515.84  6527.2  517.46  6556.6  528.26  6593.8  537.22  6751.4  540.28
#Mann= 13 ,-1 , 0
  3711.7     .05       0  4725.4      .1       0  4912.4     .12       0
  4976.9     .05       0  4995.1     .12       0  5057.2      .1       0
  5128.2     .07       0  5425.3     .12       0  5614.2     .07       0
  5953.5     .12       0  6167.4     .07       0  6440.4    .035       0
  6500.7     .05       0
Bank Sta=4976.9,4995.1
XS Rating Curve= 0 ,0
Exp/Cntr=0.3,0.1

Type RM Length L Ch R = 1 ,65164   ,742,742,742
BEGIN DESCRIPTION:
B19414
END DESCRIPTION:
XS GIS Cut Line= 3
      2325646.47      13775905.8      2324091.56     13776055.14
      2323415.13     13776819.42
#Sta/Elev= 30
  3873.5  529.97  3945.3  528.44  4327.1  508.45  4387.3  497.94  4447.6  508.04
  4477.7  500.61  4507.9  498.03  4944.5  482.38  5000.1  482.15  5010.2  481.11
  5011.1  476.12  5011.6  475.62  5029.4  476.12  5043.7  482.78  5133.2  483.26
  5241.2  482.76  5281.8  487.37  5301.5  484.52  5328.8  487.16  5379.3  497.82
  5454.2  509.23  5482.7  507.29  5588.9  514.41  5603.1  511.95  5695.1  519.22
  5709.3  516.89  5737.8  518.43  5758.7  522.26  6351.3  537.72  6456.2  538.78
#Mann= 8 ,-1 , 0
  3873.5     .05       0  4944.5      .1       0  5011.1     .05       0
  5029.4      .1       0  5043.7     .05       0  5133.2     .07       0
  5328.8    .035       0  6351.3     .07       0
Bank Sta=5011.1,5029.4
XS Rating Curve= 0 ,0
Exp/Cntr=0.3,0.1

Type RM Length L Ch R = 1 ,64422   ,504,504,504
BEGIN DESCRIPTION:
B19413
END DESCRIPTION:
XS GIS Cut Line= 3
      2324864.59     13774702.33      2324232.12     13775519.27
      2323309.88     13776687.45
#Sta/Elev= 30
  4100.9  530.38  4551.3  505.06  4800.2  504.21  4843.8  505.01  4879.1  499.68
  4943.4  482.79  4983.2  477.94  4983.9  474.13  4984.4  473.63  5002.4  474.13
  5014.8  480.68  5024.8  480.54    5307   483.3  5399.1  496.94    5428  498.82
  5442.4  494.61  5477.7  498.87  5492.1  495.03  5541.8  500.48  5556.3  497.24
  5670.1  509.32  5734.2   507.9    5848  514.83  5862.5  511.74  5912.1  516.37
  6040.4  517.17  6154.2  524.99  6218.3   523.5    6268  527.89  6622.4  535.91
#Mann= 5 ,-1 , 0
  4100.9    .035       0  4800.2     .12       0  4983.9     .05       0
  5002.4     .12       0  5024.8    .035       0
Bank Sta=4983.9,5002.4
XS Rating Curve= 0 ,0
Exp/Cntr=0.3,0.1

Type RM Length L Ch R = 1 ,63918   ,643,643,643
BEGIN DESCRIPTION:
B19412
END DESCRIPTION:
XS GIS Cut Line= 3
      2324759.19     13774561.75      2323828.02     13775211.81
      2323221.89     13776459.21
#Sta/Elev= 30
  3960.1  529.36  4014.8  527.82  4038.3  531.49  4166.6  514.65  4217.2  510.88
  4273.9  514.16  4360.2  513.54  4425.6  503.71  4446.6  503.37  4461.4  499.06
  4503.3  495.99  4562.6  498.02    4620  491.24  4742.9  484.68  4783.2  483.46
  4865.6   480.4  4948.2   478.3  4964.7  479.13  4970.8  475.64  4977.5  477.78
  4982.5  471.31    4983  470.81    5001  471.31  5006.6  479.41  5062.9  481.39
  5182.7  482.27  5365.1  490.38    5848  498.23  6163.8  509.54  6482.6  514.73
#Mann= 10 ,-1 , 0
  3960.1    .035       0    4620     .12       0  4742.9      .1       0
  4783.2     .12       0  4865.6      .1       0  4948.2     .12       0
  4982.5     .05       0    5001     .12       0  5062.9     .07       0
  5365.1     .05       0
Bank Sta=4982.5,5001
XS Rating Curve= 0 ,0
Exp/Cntr=0.3,0.1

Type RM Length L Ch R = 1 ,63275   ,581,581,581
BEGIN DESCRIPTION:
B19411
END DESCRIPTION:
XS GIS Cut Line= 4
      2324803.09     13774438.76      2323643.54     13774649.59
       2323441.5     13774921.92      2323072.55     13776318.65
#Sta/Elev= 30
  3718.7  529.71  3737.1  529.03  3747.3  532.56  3777.1   524.6  3782.2  525.84
  3835.5  507.69  3840.6  509.19  3859.1  505.43  3970.9  508.79  4000.7  502.58
  4075.7  500.03    4103  496.84  4117.6   498.9  4201.1  496.47  4311.1  490.57
  4603.6  482.93  4814.5  481.75  4942.2   476.6  4978.7  478.72  4991.4  469.74
  4991.9  469.24  5009.9  469.74  5015.3  478.46  5028.5  480.31  5134.5  479.49
    5228  478.66  5912.4  487.68    6454  500.25  6567.2  502.99    6681  506.58
#Mann= 10 ,-1 , 0
  3718.7    .035       0  4075.7     .12       0  4201.1     .07       0
  4311.1     .12       0  4603.6      .1       0  4991.4     .05       0
  5009.9      .1       0  5134.5     .05       0    6454     .07       0
  6567.2     .05       0
Bank Sta=4991.4,5009.9
XS Rating Curve= 0 ,0
Exp/Cntr=0.3,0.1

Type RM Length L Ch R = 1 ,62694   ,703,703,703
BEGIN DESCRIPTION:
Mill Creek 72.0
END DESCRIPTION:
XS GIS Cut Line= 3
      2325013.92     13774113.73      2323160.39     13774403.62
      2322879.28     13776274.76
#Sta/Elev= 30
  3001.4  521.44  3030.7  526.05  3058.8  519.49  3101.5  509.26  3111.7  502.45
    3142  506.94    3223  506.25  3273.6   503.2  3613.1   496.4  3879.6  491.47
  3901.1  482.12  3961.9   485.8  4026.8  484.15  4299.1  480.24  4424.2  478.95
  4587.3  477.76  4687.4  478.45  4815.4     478  4969.9   478.6  4990.1  477.31
  5005.8  468.17  5006.3  467.67  5024.3  468.17  5030.5  474.31    5071  477.51
  5256.1  477.12  6296.6  488.03  6624.6  495.77  6671.8   497.6  6769.6  499.32
#Mann= 14 ,-1 , 0
  3001.4     .05       0  3058.8    .035       0  3613.1     .12       0
  4026.8     .07       0  4299.1     .12       0  4424.2     .07       0
  4587.3      .1       0  4687.4     .12       0  4815.4      .1       0
  5005.8     .05       0  5024.3      .1       0  5256.1     .05       0
  6624.6     .07       0  6671.8     .05       0
Bank Sta=5005.8,5024.3
XS Rating Curve= 0 ,0
Exp/Cntr=0.3,0.1

Type RM Length L Ch R = 1 ,61991   ,557,557,557
BEGIN DESCRIPTION:
Mill Creek 71.0
END DESCRIPTION:
XS GIS Cut Line= 3
      2324978.81     13774025.88      2323134.03     13774052.23
       2321710.9     13774236.71
#Sta/Elev= 30
  3246.5  529.52  3310.3  529.15    3397  508.42  3500.3  502.39  3620.3  500.47
  3640.3  497.21  3830.4  494.29  3850.4     491  3940.4  491.44  3955.6   494.6
  3990.4  489.63  4170.6  485.88  4285.7  484.98  4670.7  478.15  4769.3  477.39
  4860.5  478.74  4966.3   476.4  4990.5  476.26  4998.3  466.01  4998.8  465.51
  5022.6  466.01  5030.5  475.25  5040.5  476.15  5199.9  477.29    5272  477.03
    5393  482.53    5801  494.12  5991.6  500.56  6360.1  514.31  6526.5  519.78
#Mann= 14 ,-1 , 0
  3246.5     .05       0    3397    .035       0  3955.6     .12       0
  4170.6    .035       0  4285.7     .07       0  4670.7    .035       0
  4769.3     .07       0  4966.3      .1       0  4998.3     .05       0
  5022.6      .1       0  5199.9     .07       0    5801    .035       0
  5991.6     .05       0  6360.1    .035       0
Bank Sta=4998.3,5022.6
XS Rating Curve= 0 ,0
Exp/Cntr=0.3,0.1

Type RM Length L Ch R = 1 ,61434   ,484,484,484
BEGIN DESCRIPTION:
Mill Creek 70.0
END DESCRIPTION:
XS GIS Cut Line= 3
      2325040.34     13773929.25      2323213.09     13773525.15
      2321710.92      13773551.5
#Sta/Elev= 30
  3040.1  527.03  3082.2  528.35  3137.7  526.52  3218.2  508.08  3387.8  503.21
  3660.1  497.16  3777.7  496.46  3803.4  493.75  4334.9  486.61  4403.6  484.02
  4588.4  478.29  4609.3  476.49  4760.2  474.34  4880.9  475.79  4969.6   476.3
  4979.6  474.66  4987.5  464.86    4988  464.36  5011.8  464.86  5019.6  476.15
  5033.5  476.06  5143.3  474.82  5249.6   476.5  5289.6  479.23  5459.7  480.62
  5822.2  488.86  6032.5  492.46  6229.6  496.27  6353.6  498.98  6413.9  500.05
#Mann= 15 ,-1 , 0
  3040.1     .05       0  3387.8    .035       0  4334.9     .07       0
  4403.6    .035       0  4588.4     .07       0  4760.2      .1       0
  4880.9    .035       0  4987.5    .035       0  5011.8    .035       0
  5033.5      .1       0  5143.3     .07       0  5822.2    .035       0
  6032.5     .07       0  6229.6     .05       0  6353.6     .07       0
Bank Sta=4987.5,5011.8
XS Rating Curve= 0 ,0
Exp/Cntr=0.3,0.1

Type RM Length L Ch R = 1 ,60950   ,559,559,559
BEGIN DESCRIPTION:
Mill Creek 69.0
END DESCRIPTION:
XS GIS Cut Line= 3
      2324583.49     13773270.39        2323125.       13773075.
      2321491.26     13773138.62
#Sta/Elev= 30
  3528.8  502.18    3691  497.96  3913.3  491.45  4074.2  488.62  4526.1  485.41
  4556.4  483.89  4576.6   480.5  4583.9  483.63  4596.7  484.33  4788.3   481.1
  4890.9  477.69  4929.7  474.43  4970.1  474.28  4990.2  470.89  4997.8  466.54
  4998.1   462.3  4998.6   461.8  5022.6   462.3  5030.3  472.94  5060.4  475.06
  5280.5  474.67  5390.7  480.39  5590.8  480.07  5660.8  476.81  5730.9  480.62
  6141.2  485.65  6151.2  486.01  6161.5  489.22  6211.2  490.91  6635.3  496.13
#Mann= 7 ,-1 , 0
  3528.8     .07       0    3691    .035       0  3913.3     .05       0
  4074.2     .07       0  4788.3    .035       0  4998.1    .035       0
  5022.6    .035       0
Bank Sta=4998.1,5022.6
XS Rating Curve= 0 ,0
Exp/Cntr=0.3,0.1

Type RM Length L Ch R = 1 ,60391   ,552,552,552
BEGIN DESCRIPTION:
Mill Creek 68.0
END DESCRIPTION:
XS GIS Cut Line= 3
      2324513.25     13772883.87        2322825.       13772625.
      2321429.89     13772883.85
#Sta/Elev= 30
  3297.2  499.68  3558.5  489.67  3922.7  485.79  4380.7  484.78  4570.2  480.03
  4707.5  474.84  4775.9  473.32  4814.9  474.01  4964.7  474.84    4971   472.4
    4976  473.81  4982.8  462.28  4983.3  461.78  5007.4  462.28  5007.7  466.08
  5015.3  473.85  5025.5  474.68  5087.2  472.26  5178.1  474.85  5381.5  475.45
  5585.4  480.39  5633.1   482.7  5928.3  486.75  5977.5  487.59  6160.5  489.33
  6181.8  489.01  6186.9  490.16  6234.6  488.89  6297.6  491.84  6424.1  492.14
#Mann= 8 ,-1 , 0
  3297.2     .05       0  4814.9      .1       0  4982.8     .05       0
  5007.4      .1       0  5087.2     .07       0  5928.3     .05       0
  5977.5    .035       0  6160.5    .063       0
Bank Sta=4982.8,5007.4
XS Rating Curve= 0 ,0
Exp/Cntr=0.3,0.1

Type RM Length L Ch R = 1 ,59839   ,516,516,516
BEGIN DESCRIPTION:
Mill Creek 67.0
END DESCRIPTION:
XS GIS Cut Line= 3
      2324293.57     13771706.73      2322817.78     13772207.45
      2321201.41     13772822.37
#Sta/Elev= 30
  3591.7  500.68  3596.3  500.37  4037.8  480.74  4075.9  478.44  4101.1  480.54
  4234.1  479.35    4466  483.13  4519.5  483.86    4594  481.63  4766.8  476.05
  4865.6  474.23  4940.9  472.92  4984.1  473.61  4988.9  460.48  4989.4  459.98
  5013.5  460.48  5032.6  473.77  5152.1  473.51  5253.3  472.91  5327.8  472.04
  5436.6  477.36  5559.7  481.59  5892.6   483.4  6005.2  483.62  6148.1  481.84
  6212.3  483.29    6367  485.52  6425.4  484.49  6615.9  488.97  6879.5  494.83
#Mann= 19 ,-1 , 0
  3591.7     .05       0  3596.3     .07       0  4037.8     .12       0
  4234.1     .07       0    4466     .12       0    4594     .07       0
  4766.8     .05       0  4865.6     .07       0  4940.9      .1       0
  4988.9     .05       0  5013.5      .1       0  5152.1     .12       0
  5253.3     .07       0  5436.6     .05       0  5892.6     .07       0
  6005.2     .05       0  6212.3    .035       0  6425.4     .05       0
  6615.9    .035       0
Bank Sta=4988.9,5013.5
XS Rating Curve= 0 ,0
Exp/Cntr=0.3,0.1

Type RM Length L Ch R = 1 ,59323   ,650,650,650
BEGIN DESCRIPTION:
Mill Creek 66.0
END DESCRIPTION:
XS GIS Cut Line= 3
      2323880.75     13771285.04        2322675.       13771775.
      2321113.54     13772629.12
#Sta/Elev= 30
  3702.6  495.82  3914.4   488.4  4205.3  476.53  4421.2  473.27  4518.4  474.36
  4804.6  471.55  4873.4  472.47  4965.3  472.67  4971.7  471.32  4982.4  460.63
  4982.9  460.13  5007.1  460.63  5012.2  470.74  5017.9  472.76  5055.8  470.66
  5071.9  472.17  5099.4  470.57  5162.6  471.69  5209.3  473.04  5330.8  471.55
  5390.8  472.46  6127.6  477.72  6264.2  480.15  6307.8  483.02    6324  482.23
  6329.7  483.87  6367.6  482.07  6417.5  483.92  6668.2  491.93  6783.9  493.59
#Mann= 10 ,-1 , 0
  3702.6     .05       0  3914.4     .07       0  4873.4      .1       0
  4982.4     .05       0  5007.1      .1       0  5162.6     .12       0
  5330.8     .07       0  5390.8     .05       0  6127.6     .07       0
  6417.5     .05       0
Bank Sta=4982.4,5007.1
XS Rating Curve= 0 ,0
Exp/Cntr=0.3,0.1

Type RM Length L Ch R = 1 ,58673   ,490,490,490
BEGIN DESCRIPTION:
B19410
END DESCRIPTION:
XS GIS Cut Line= 4
      2323696.26     13771065.44      2322457.61     13771267.48
      2322264.35      13771258.7      2320612.85     13771162.07
#Sta/Elev= 30
  3673.8  490.81  3728.7  489.19  3959.2  482.48    4010  481.77  4252.6  480.27
  4330.3  477.19  4430.6  474.19  4546.4  470.55  4622.3  470.21  4831.6  471.29
  4971.5   471.9  4981.5  471.03  4991.5  467.33  4997.9  459.93  4998.4  459.43
  5025.2  459.93  5030.3  467.98  5031.5  469.88  5041.5  471.19  5071.6  470.68
  5081.6  468.72  5090.1   469.8  5095.1  467.76  5101.6  469.69  5128.7  470.52
  5642.5  475.79  5822.8  480.28  6023.2  489.27  6353.7  490.65  6776.6  506.63
#Mann= 12 ,-1 , 0
  3673.8     .05       0  3728.7     .07       0  3959.2     .05       0
    4010     .07       0  4330.3     .05       0  4430.6     .07       0
  4622.3     .05       0  4831.6      .1       0  4997.9     .05       0
  5025.2      .1       0  5030.3     .07       0  5128.7     .05       0
Bank Sta=4997.9,5025.2
XS Rating Curve= 0 ,0
Exp/Cntr=0.3,0.1

Type RM Length L Ch R = 1 ,58183   ,556,556,556
BEGIN DESCRIPTION:
Mill Creek 65.0
END DESCRIPTION:
XS GIS Cut Line= 3
      2323524.97       13770875.        2322425.       13770825.
      2320824.97     13769524.97
#Sta/Elev= 30
  3898.9   490.4    3900   490.4  3937.8  489.56  4038.1  485.82  4221.5  481.96
  4329.3  481.33  4559.5  473.56  4839.1  468.49    4980  470.89    4990  467.11
  4993.5  460.31    4994  459.81  5020.8  460.31  5021.6  469.83  5070.3  470.06
  5120.7  469.41  5194.2  466.37  5282.6  468.56  5318.2  468.81  5440.3  467.41
  5957.8   472.2  6061.7  476.32  6092.3   477.5  6159.4  481.12  6309.6   497.1
    6546  507.26    6813  514.16  6902.1  518.49  7053.1  528.59  7061.6   529.3
#Mann= 20 ,-1 , 0
  3898.9     .07       0    3900     .05       0  3937.8     .07       0
  4038.1     .05       0  4221.5     .07       0  4839.1      .1       0
  4993.5     .05       0  5020.8      .1       0  5070.3     .07       0
  5120.7      .1       0  5194.2     .05       0  5282.6      .1       0
  5318.2     .07       0  5957.8     .12       0  6061.7     .07       0
  6092.3     .12       0  6309.6     .07       0    6546     .05       0
  6902.1     .07       0  7053.1     .05       0
Bank Sta=4993.5,5020.8
XS Rating Curve= 0 ,0
Exp/Cntr=0.3,0.1

Type RM Length L Ch R = 1 ,57627   ,531,531,531
BEGIN DESCRIPTION:
Mill Creek 64.0
END DESCRIPTION:
XS GIS Cut Line= 3
      2323475.01       13770825.        2322375.       13770325.
      2321674.97     13769674.98
#Sta/Elev= 30
  3772.8  489.77  3805.6  488.98  3882.2  486.03  3992.5   482.8  4050.2   482.7
  4270.4  481.24  4552.7  471.69  4725.4  467.67  4776.8  468.07  4828.4  465.92
    4846  467.93  4984.5  469.94  4988.2  469.24  4988.6  462.15  4989.1  461.65
  5016.1  462.15  5037.5  462.71  5044.9  467.24  5051.7  465.21  5059.1  469.86
    5231  467.26  5299.4  465.77  5306.8  467.11  5455.3  467.81  5542.6   478.1
  5667.4  492.05  5829.6  500.94  5858.4  504.81  5885.1  506.46  5936.4  510.12
#Mann= 11 ,-1 , 0
  3772.8     .05       0  3805.6     .07       0  3882.2     .05       0
  4050.2     .07       0  4725.4      .1       0  4988.6     .05       0
  5016.1      .1       0    5231     .07       0  5542.6     .12       0
  5829.6    .035       0  5885.1     .07       0
Bank Sta=4988.6,5016.1
XS Rating Curve= 0 ,0
Exp/Cntr=0.3,0.1

Type RM Length L Ch R = 1 ,57096   ,540,540,540
BEGIN DESCRIPTION:
Mill Creek 63.0
END DESCRIPTION:
XS GIS Cut Line= 3
        2323575.       13770825.        2322475.       13769875.
      2322124.96     13769674.98
#Sta/Elev= 30
  3540.5  491.23  3577.4  491.56  3595.1  491.02  3809.6  484.74    3958  481.49
    4242  480.81  4650.7  467.67  4738.9  469.27  4873.8  467.13  4880.4  469.81
  4888.1  467.62  4894.7  471.53  4901.4  468.87  4918.2  472.54  4937.4  473.16
    4944   468.6  4958.3  467.33  4965.9  469.41  4972.6  467.01  4986.8  467.71
  4988.1  463.79  4988.6  463.29  5015.7  463.79  5119.9  467.73  5155.2  466.16
  5163.1   467.3  5190.5  481.76  5219.6  485.82  5305.3   490.9  5397.1  493.74
#Mann= 11 ,-1 , 0
  3540.5     .07       0  3577.4     .05       0  3595.1     .07       0
  3809.6     .05       0    3958     .07       0  4650.7      .1       0
  4918.2    .035       0  4988.1    .035       0  5015.7    .035       0
  5219.6    .063       0  5305.3    .035       0
Bank Sta=4988.1,5015.7
XS Rating Curve= 0 ,0
Exp/Cntr=0.3,0.1

Type RM Length L Ch R = 1 ,56556   ,550,550,550
BEGIN DESCRIPTION:
Mill Creek 62.0
END DESCRIPTION:
XS GIS Cut Line= 3
      2323525.02     13770625.03        2322725.       13769525.
      2322024.98       13769375.
#Sta/Elev= 30
  3639.4  488.91  3687.3  487.38  3748.5   485.7  3829.2  483.67  3893.7  482.29
  4004.2  480.52  4289.7  477.26  4347.7  478.32    4398  472.05  4557.9  476.46
  4705.5  476.85    4777  469.96  4820.7  472.72  4898.4  466.57  4971.4   465.1
  4972.2  462.46  4972.7  461.96    5000  462.46  5060.9   462.8  5091.6  467.35
  5222.3  474.74  5243.7  475.95  5347.3  480.52  5360.1   476.8  5388.2  476.93
  5404.4  478.31  5409.5  483.39  5418.9  484.49  5622.7  499.99  5715.5  508.89
#Mann= 14 ,-1 , 0
  3639.4     .05       0  3687.3     .07       0  3748.5     .05       0
  3829.2     .07       0  3893.7     .05       0  4004.2     .07       0
  4289.7    .035       0  4557.9    .063       0  4898.4      .1       0
  4972.2     .05       0    5000      .1       0  5222.3    .035       0
  5243.7     .12       0  5622.7    .035       0
Bank Sta=4972.2,5000
XS Rating Curve= 0 ,0
Exp/Cntr=0.3,0.1

Type RM Length L Ch R = 1 ,56006   ,540,540,540
BEGIN DESCRIPTION:
Mill Creek 61.0
END DESCRIPTION:
XS GIS Cut Line= 3
      2323974.98     13770124.98        2322875.       13769025.
        2322375.       13768725.
#Sta/Elev= 30
  3444.4  486.75  3557.5  484.59  3599.9  482.26  3614.1  489.71  3621.1  490.37
  3670.6  486.33  3739.3  484.09  3840.3  483.16  3863.5  480.01  3882.8   479.2
  3899.1  482.23  3911.1  482.66  3939.3  479.82  3998.8  479.34  4391.9   477.1
  4654.5  468.97  4745.4  465.57  4985.9  467.46  4996.5  463.36  4999.7  458.31
  5000.2  457.81  5027.5  458.31    5035  467.83  5067.7  466.42  5108.8  466.02
  5161.3     470  5233.2  477.13  5400.4  489.33  5451.3  495.77  5583.1  507.09
#Mann= 10 ,-1 , 0
  3444.4    .094       0  3739.3     .07       0  3863.5    .035       0
  3899.1     .05       0  3998.8     .07       0  4654.5      .1       0
  4999.7     .05       0  5027.5      .1       0  5067.7     .12       0
  5451.3     .07       0
Bank Sta=4999.7,5027.5
XS Rating Curve= 0 ,0
Exp/Cntr=0.3,0.1

Type RM Length L Ch R = 1 ,55466   ,564,564,564
BEGIN DESCRIPTION:
Mill Creek 60.0
END DESCRIPTION:
XS GIS Cut Line= 3
      2323874.99     13769924.98        2323225.       13768675.
      2322974.99     13768274.98
#Sta/Elev= 30
  3587.1  491.37  3609.6  489.64  3617.4  486.36  3623.1  487.05  3639.5  480.81
  3683.7   478.9    3742  479.57  3944.1  479.61  4169.4  478.21  4197.8  477.66
  4449.6  473.19  4452.1  473.03  4669.1  471.51  4810.9  465.54  4886.5  464.99
  4928.3  466.58  5009.5  466.25    5011  456.83  5011.5  456.33  5038.8  456.83
  5040.2  465.49  5054.9  467.01  5074.5  465.43  5113.3  465.67  5182.2  470.63
  5192.7  470.91    5311  483.62  5351.9  488.81  5417.6  498.07  5467.7  500.26
#Mann= 15 ,-1 , 0
  3587.1     .07       0    3742     .05       0  3944.1     .07       0
  4169.4     .12       0  4197.8     .07       0  4449.6     .12       0
  4452.1     .07       0  4886.5      .1       0    5011     .05       0
  5038.8      .1       0  5074.5     .12       0  5182.2     .07       0
  5192.7    .035       0    5311     .07       0  5351.9    .035       0
Bank Sta=5011,5038.8
XS Rating Curve= 0 ,0
Exp/Cntr=0.3,0.1

Type RM Length L Ch R = 1 ,54902   ,625,625,625
BEGIN DESCRIPTION:
Mill Creek 59.0
END DESCRIPTION:
XS GIS Cut Line= 3
      2324625.01     13769925.02        2323675.       13768375.
        2323475.       13768025.
#Sta/Elev= 30
  3185.6  495.42  3382.9   490.2  3678.8  477.69  3773.6  472.41  3804.5   472.1
  3905.1  475.34  4204.8  468.14  4500.8  466.32    4590   464.3  4616.8  464.22
    4640  461.95  4675.2     462  4707.5  464.61  4779.2  465.16  4815.9  462.75
    4932  465.49  4980.4  465.03  4986.7  457.81  4987.2  457.31  5014.6  457.81
  5017.3  461.54  5026.6  464.38  5118.9  471.94  5151.2  476.11  5237.5  483.39
    5275  489.23  5296.6  490.37  5312.4  493.78  5394.4  496.13  5406.7  496.15
#Mann= 7 ,-1 , 0
  3185.6     .05       0    4590     .12       0  4707.5      .1       0
  4986.7     .05       0  5014.6      .1       0  5118.9     .12       0
  5394.4     .07       0
Bank Sta=4986.7,5014.6
XS Rating Curve= 0 ,0
Exp/Cntr=0.3,0.1

Type RM Length L Ch R = 1 ,54277   ,723,723,723
BEGIN DESCRIPTION:
B19409
END DESCRIPTION:
XS GIS Cut Line= 3
      2324803.14     13769818.05      2324205.76     13768315.83
      2323652.91      13767859.5
#Sta/Elev= 30
  3552.4  491.22  3728.3  488.47  3992.7  476.56  4316.5  468.47  4470.4   465.5
  4801.5   463.2  4868.6  463.43  4891.2  461.76  4924.9  463.84    4987  464.55
  4994.6  457.21  4995.1  456.71  5022.5  457.21  5023.5   460.7    5030   464.6
  5077.4  464.31  5107.1     462  5139.3  465.75  5142.6  466.29  5166.8  470.15
  5269.9  480.01  5319.4  481.98  5354.5   480.8  5432.7  483.72  5475.7  486.93
  5660.7  491.05  5774.1  491.37  5823.6  489.41  5852.2  490.82  5885.9  488.85
#Mann= 7 ,-1 , 0
  3552.4     .05       0  4801.5     .07       0  4924.9      .1       0
  4994.6     .05       0  5022.5      .1       0  5139.3     .12       0
  5142.6     .07       0
Bank Sta=4994.6,5022.5
XS Rating Curve= 0 ,0
Exp/Cntr=0.3,0.1

Type RM Length L Ch R = 1 ,53554   ,657,657,657
BEGIN DESCRIPTION:
B19408
END DESCRIPTION:
XS GIS Cut Line= 3
       2325857.3      13769431.5      2324697.71     13768394.89
      2323731.41     13767797.55
#Sta/Elev= 30
  3627.8  494.16    3740  492.88  3792.2  490.78  3839.4  489.04  4055.6  481.51
  4110.1  479.27  4526.6  466.89  4813.2  463.91  4894.4  461.29  4955.8  462.65
  4965.5  463.44  4972.2  461.49  5000.6  458.88  5000.8  456.92  5001.3  456.42
  5028.9  456.92    5029  461.41  5050.7  463.49  5160.7  463.85  5271.8  462.02
  5329.5  463.85  5439.4  462.71  5515.3  463.94  5681.4  466.86  5765.7  468.91
  5920.2  477.75  6028.1  484.75  6051.4  484.94  6180.6  487.05  6319.2  485.91
#Mann= 15 ,-1 , 0
  3627.8     .05       0  3792.2     .07       0  3839.4     .05       0
  4055.6     .07       0  4110.1     .05       0  4813.2     .12       0
  4955.8      .1       0  5000.8     .05       0  5028.9      .1       0
  5160.7     .12       0  5271.8      .1       0  5515.3     .12       0
  5681.4     .07       0  5920.2     .05       0  6051.4     .07       0
Bank Sta=5000.8,5028.9
XS Rating Curve= 0 ,0
Exp/Cntr=0.3,0.1

Type RM Length L Ch R = 1 ,52897   ,724,724,724
BEGIN DESCRIPTION:
B19407
END DESCRIPTION:
XS GIS Cut Line= 4
      2326059.35     13769167.96      2325461.97     13768175.27
      2324706.49     13767797.53      2323618.63     13767674.71
#Sta/Elev= 30
  3353.1  491.74  3778.8   487.4  3903.2   483.3  4029.1  476.58  4173.5   472.4
  4511.7  474.73  4689.7  471.21  4795.5  467.12    4904  459.61  4933.1  462.65
  4960.6  462.67  4993.8   462.9  5000.2  458.87  5002.1  454.73  5002.6  454.23
  5030.3  454.73    5033  462.32  5105.6  460.41  5167.1  463.11  5229.5  462.54
    5338  462.74  5438.5  462.36  5537.2  462.79    5636  463.51  6052.2  476.64
  6122.7  480.04  6203.2  481.28  6311.8   482.4  6354.3  481.06  6451.1  481.42
#Mann= 16 ,-1 , 0
  3353.1     .05       0  3778.8     .07       0  3903.2     .05       0
  4689.7     .07       0  4795.5     .12       0    4904      .1       0
  4960.6     .12       0  5002.1     .05       0  5030.3     .12       0
  5229.5     .07       0    5338     .05       0  5438.5     .07       0
  5537.2     .12       0    5636     .05       0  6052.2     .07       0
  6354.3    .035       0
Bank Sta=5002.1,5030.3
XS Rating Curve= 0 ,0
Exp/Cntr=0.3,0.1

Type RM Length L Ch R = 1 ,52173   ,829,829,829
BEGIN DESCRIPTION:
Mill Creek 58.0
END DESCRIPTION:
XS GIS Cut Line= 3
      2326103.23     13769097.62      2325224.79     13767305.59
       2324636.2     13765592.54
#Sta/Elev= 30
  3094.3  489.83  3512.7  484.02  3737.7  474.77  3855.7  472.38  4007.6  472.47
  4170.7  474.78  4401.2  474.39    4694  463.28  4773.7  462.03  4845.6  459.39
  4957.1  462.43  4969.2  460.83    4972   453.6  4972.5   453.1  5000.2   453.6
  5001.6  461.39  5106.4  462.09  5230.7  463.22  5577.1  461.72  6137.5  463.18
    6246  464.71  6402.2  469.48  6428.2  470.64  6468.7  475.67  6641.6   491.8
  6646.9  491.17  6756.6   500.1  6797.9  502.75  6893.8  514.41  6901.4  515.23
#Mann= 9 ,-1 , 0
  3094.3     .05       0    4694     .07       0  4773.7      .1       0
    4972     .05       0  5000.2      .1       0  5106.4     .05       0
  6468.7     .07       0  6756.6     .12       0  6893.8    .035       0
Bank Sta=4972,5000.2
XS Rating Curve= 0 ,0
Exp/Cntr=0.3,0.1

Type RM Length L Ch R = 1 ,51344   ,928,928,928
BEGIN DESCRIPTION:
Mill Creek 57.0
END DESCRIPTION:
XS GIS Cut Line= 3
      2327087.15     13768719.94      2326024.19     13767226.53
      2325716.73     13765662.85
#Sta/Elev= 30
  3226.1  499.57  3410.5  492.93  3639.8  480.57  3687.6  478.75  3754.8  473.63
  3848.3  471.05    4131  465.52  4902.9   460.2  4949.8  460.73  4987.4  460.28
  4995.5  455.45  5001.6  456.25  5002.3  452.33  5002.8  451.83  5030.5  452.33
  5031.1  459.86  5045.9  461.21  5181.6  459.79  5232.6   457.7  5295.1  461.16
  5795.7   458.3  5976.7  462.15    6173  469.34  6270.1  478.63  6378.8  489.45
    6406  497.95    6430  495.86  6530.5  500.75  6542.7  500.35  6652.8  501.31
#Mann= 16 ,-1 , 0
  3226.1    .035       0  3639.8     .12       0  3687.6    .035       0
  3848.3     .07       0    4131     .05       0  4902.9     .07       0
  4949.8     .12       0  5002.3     .05       0  5030.5     .12       0
  5181.6     .05       0  5795.7     .07       0  5976.7     .05       0
  6270.1     .07       0  6378.8     .12       0  6530.5     .07       0
  6542.7     .12       0
Bank Sta=5002.3,5030.5
XS Rating Curve= 0 ,0
Exp/Cntr=0.3,0.1

Type RM Length L Ch R = 1 ,50416   ,447,447,447
BEGIN DESCRIPTION:
Mill Creek 56.0
END DESCRIPTION:
XS GIS Cut Line= 3
      2327315.55     13768588.19        2326725.       13766725.
      2326474.98     13766374.97
#Sta/Elev= 30
    3050  495.97  3210.8  489.51  3217.5  489.27  3312.8  485.24  3421.3  481.51
  3447.8  480.66  3466.6   480.8  3483.4  476.55  3493.7  478.37  3525.4  475.06
  3682.8  474.01  3968.4  468.78  4083.7   465.7  4342.7  461.68  4595.7  458.02
  4668.9  460.19  4878.7  458.86  4950.9  460.23    4963  457.75  4973.1   456.9
  4978.9  454.07  4979.4  453.57  5009.3  454.07  5011.9  456.86  5026.7   458.3
  5104.6  461.07  5228.1  470.81  5331.5  479.07  5351.7  480.98  5434.7  487.51
#Mann= 16 ,-1 , 0
    3050     .07       0  3210.8     .05       0  3217.5     .12       0
  3312.8    .035       0  3421.3     .05       0  3447.8     .07       0
  3968.4     .05       0  4083.7     .07       0  4342.7    .035       0
    4963     .05       0  4978.9     .05       0  5009.3     .05       0
  5104.6     .12       0  5228.1     .07       0  5331.5     .12       0
  5351.7     .07       0
Bank Sta=4978.9,5009.3
XS Rating Curve= 0 ,0
Exp/Cntr=0.3,0.1

Type RM Length L Ch R = 1 ,49969   ,627,627,627
BEGIN DESCRIPTION:
Mill Creek 55.0
END DESCRIPTION:
XS GIS Cut Line= 3
      2327860.18     13768289.45      2327148.63      13766725.8
      2327034.43     13765961.52
#Sta/Elev= 30
  3137.3  499.01  3177.3  496.86  3229.4   495.9  3286.6  492.17  3648.9  477.14
  3913.5  470.92    4098  468.41  4149.6  465.84  4267.7  464.86  4494.4  463.46
  4592.4  458.56  4632.8  457.73  4647.4  456.23  4665.5  457.25  4821.4   458.5
  4924.4  459.71  4936.9  459.61    4947  458.13  4957.2  454.51  4961.6  450.34
  4962.1  449.84    4992  450.34  4997.6  455.55  5007.7  458.55  5024.3  460.75
  5124.3  464.65  5230.1  468.39  5280.7   468.5  5432.4  474.94    5628  478.55
#Mann= 10 ,-1 , 0
  3137.3    .035       0  3177.3     .05       0  4267.7     .07       0
  4665.5     .12       0  4821.4     .07       0  4924.4     .12       0
  4961.6     .05       0    4992     .12       0  5024.3     .07       0
  5124.3     .05       0
Bank Sta=4961.6,4992
XS Rating Curve= 0 ,0
Exp/Cntr=0.3,0.1

Type RM Length L Ch R = 1 ,49342   ,535,535,535
BEGIN DESCRIPTION:
Mill Creek 54.0
END DESCRIPTION:
XS GIS Cut Line= 3
      2327924.99     13767124.99        2327625.       13766725.
        2327425.     13766374.99
#Sta/Elev= 30
    4500  475.37    4600   470.1  4613.5  470.27  4657.3  467.22  4778.1  463.37
  4842.7  463.57  4865.5  461.45  4886.4  459.88  4928.1  459.03  4942.3  457.01
    4950   456.1  4986.4  457.29  4992.5  448.04    4993  447.54  5023.3  448.04
  5029.5  458.08  5093.8  457.14  5153.3  455.95  5190.7  463.46  5196.5  463.28
  5206.6  466.29  5228.2  469.18  5233.9  468.94  5287.2  473.15    5293  472.51
  5308.8  474.67  5336.1  475.19  5354.6   477.3  5367.8  478.31  5403.1  478.56
#Mann= 7 ,-1 , 0
    4500     .05       0  4865.5     .07       0  4942.3     .12       0
  4992.5     .05       0  5023.3     .12       0  5093.8      .1       0
  5354.6     .05       0
Bank Sta=4992.5,5023.3
XS Rating Curve= 0 ,0
Exp/Cntr=0.3,0.1

Type RM Length L Ch R = 1 ,48807   ,544,544,544
BEGIN DESCRIPTION:
Mill Creek 53.0
END DESCRIPTION:
XS GIS Cut Line= 3
      2328325.02     13766925.04        2328075.       13766475.
      2327575.04     13766325.01
#Sta/Elev= 30
    4481  474.26  4494.8  473.58  4510.8  471.64  4554.3   469.5    4584   466.9
  4760.2  458.63  4781.9  456.92    4870  455.79  4906.6  457.21  4998.4  457.49
  5002.2  447.01  5002.7  446.51  5032.5  446.51    5033  447.01  5037.6  454.46
  5045.4  456.73  5083.7  456.08  5149.8  456.63    5155  456.03  5162.9  453.93
  5182.9  452.71  5193.7  456.65  5221.2  457.47  5246.4  459.13  5254.2  458.81
  5342.8  465.08  5358.6  466.82    5430  471.21  5484.9  473.02  5517.8  474.61
#Mann= 6 ,-1 , 0
    4481     .07       0  5002.2     .05       0    5033     .07       0
  5193.7    .035       0  5342.8      .1       0  5484.9     .05       0
Bank Sta=5002.2,5033
XS Rating Curve= 0 ,0
Exp/Cntr=0.3,0.1
