HEC-RAS study NASH CREEK.prj: NASH CREEK Base Level Engineering

--- NASH CREEK.g01 (geometry) --- (continued)

Type RM Length L Ch R = 1 ,56231   ,475,475,475
BEGIN DESCRIPTION:
NASH CREEK 92.0
END DESCRIPTION:
XS GIS Cut Line= 3
      2357374.98     13770674.96        2357225.       13770325.
      2356674.99     13769724.99
#Sta/Elev= 30
    4625  508.15  4722.9  504.11  4755.5  504.93  4838.9   501.2  4844.4  499.56
  4862.5  499.36  4867.9  497.78  4886.1  496.94  4896.9  494.15  4915.1  493.42
  4920.5  491.49  4924.2  491.51  4938.6  490.93  4944.1  488.38  4953.9  487.58
  4954.4  487.08  4970.5  487.58  4991.2  488.15  5019.6  492.29  5055.4  492.61
  5076.3  495.68  5118.2  496.72    5166   497.3  5387.7  498.79  5635.6   503.7
  5784.2  507.46  5798.4  508.42  5805.8  509.48  5812.6  512.16  5819.7   512.4
#Mann= 6 ,-1 , 0
    4625     .07       0  4924.2     .12       0  4953.9     .05       0
  4970.5     .12       0  5118.2      .1       0    5166     .07       0
Bank Sta=4953.9,4970.5
XS Rating Curve= 0 ,0
Exp/Cntr=0.3,0.1

Type RM Length L Ch R = 1 ,55756   ,442,442,442
BEGIN DESCRIPTION:
NASH CREEK 91.0
END DESCRIPTION:
XS GIS Cut Line= 3
        2357825.     13770725.01        2357625.       13770125.
      2357124.99     13769524.99
#Sta/Elev= 30
  4372.1  511.04  4414.3   509.6  4452.5  506.43  4455.1  506.24    4604  502.55
  4656.7   502.3  4867.5  496.21  4920.2  495.28  4951.9  496.16  4972.9  494.09
  4983.5  488.37  4990.7  486.98  5003.4   485.8  5003.9   485.3  5020.1   485.8
  5026.8  489.29    5069  492.83  5147.1   493.8  5196.6  492.39  5252.5  494.53
  5271.9  494.06  5352.8  494.78  5367.1   495.3  5395.1   498.6  5420.5  498.92
  5451.7  498.06  5537.6  500.39  5558.4  501.94  5665.2  503.68  5785.6  507.74
#Mann= 9 ,-1 , 0
  4372.1     .07       0  4452.5     .12       0  4455.1     .07       0
  4990.7     .12       0  5003.4     .05       0  5020.1     .12       0
  5026.8      .1       0  5271.9     .12       0  5420.5     .07       0
Bank Sta=5003.4,5020.1
XS Rating Curve= 0 ,0
Exp/Cntr=0.3,0.1

Type RM Length L Ch R = 1 ,55314   ,450,450,450
BEGIN DESCRIPTION:
NASH CREEK 90.0
END DESCRIPTION:
XS GIS Cut Line= 3
        2357875.     13770774.99        2357975.       13769875.
      2357424.98     13769274.98
#Sta/Elev= 30
  4099.3  514.42  4237.7  508.41  4280.4  503.87  4461.5  500.34  4602.4  495.96
  4709.2  494.48  4843.8  493.78    4874  492.11  4894.1  493.23  4919.7  491.76
  4954.5  486.37  4994.8  488.36  5010.3  486.29  5010.8  485.79    5027  486.29
  5032.9  488.99  5047.1  490.12  5103.8  490.67  5214.2  494.78    5274  494.76
  5386.8  498.39    5451  498.57  5521.2  501.48  5592.2  501.76  5626.9  503.15
  5712.4  506.11  5782.9  515.13  5811.7  517.07  5815.4  518.94  5818.8  518.94
#Mann= 9 ,-1 , 0
  4099.3     .12       0  4237.7     .07       0  4709.2     .12       0
  4919.7      .1       0  5010.3     .05       0    5027      .1       0
  5214.2     .12       0  5626.9     .07       0  5782.9     .12       0
Bank Sta=5010.3,5027
XS Rating Curve= 0 ,0
Exp/Cntr=0.3,0.1

Type RM Length L Ch R = 1 ,54864   ,389,389,389
BEGIN DESCRIPTION:
NASH CREEK 89.0
END DESCRIPTION:
XS GIS Cut Line= 3
      2357975.01     13770724.98        2358375.       13769925.
        2358375.     13769325.01
#Sta/Elev= 30
  4110.8  513.75  4147.1  511.94  4155.5  512.91  4169.5  510.73  4223.2  507.75
  4275.7  503.37  4370.7  502.11  4585.7  495.58  4887.6   489.8  4929.7  490.43
  4968.9  485.02    4996  486.19  5015.2  485.51  5075.2   491.6  5095.2  489.79
  5125.2     491  5187.7  489.13  5215.2  487.36  5235.2  483.54  5275.2  485.43
  5296.8  482.19  5297.3  481.69  5313.6  482.19  5325.2  486.09  5345.2  488.35
  5355.2  492.57  5365.2  494.19    5475  500.08  5587.5  508.48  5605.2  510.25
#Mann= 10 ,-1 , 0
  4110.8     .12       0  4223.2     .07       0  4585.7     .12       0
  4887.6      .1       0    4996     .12       0  5187.7      .1       0
  5296.8     .05       0  5313.6      .1       0    5475     .07       0
  5587.5     .12       0
Bank Sta=5296.8,5313.6
XS Rating Curve= 0 ,0
Exp/Cntr=0.3,0.1

Type RM Length L Ch R = 1 ,54475   ,484,484,484
BEGIN DESCRIPTION:
B19769
END DESCRIPTION:
XS GIS Cut Line= 3
      2358579.94     13770729.65      2358601.05     13769948.44
       2358442.7     13769251.71
#Sta/Elev= 30
  4415.3  516.95    4520   509.5    4570  503.28  4713.4  496.43  4780.1  489.12
  4786.4  490.78  4791.4  489.12  4811.8  487.87  4830.1   486.3  4920.1  485.93
  4990.2  482.71  5030.2  485.79  5070.2  486.26  5100.2  484.64  5130.2  485.95
  5180.2  485.31  5187.6  482.24  5188.1  481.74  5204.5  482.24  5231.1   486.1
  5395.2  488.37  5436.2  486.72  5456.7  487.27    5467  488.64  5472.2  490.74
  5604.7  493.21  5713.1   498.2  5815.3  507.17  5875.2  514.36  5911.3  516.94
#Mann= 7 ,-1 , 0
  4415.3     .07       0  4713.4     .12       0  4811.8      .1       0
  5187.6     .05       0  5204.5      .1       0  5604.7     .07       0
  5815.3     .12       0
Bank Sta=5187.6,5204.5
XS Rating Curve= 0 ,0
Exp/Cntr=0.3,0.1

Type RM Length L Ch R = 1 ,53991   ,438,438,438
BEGIN DESCRIPTION:
NASH CREEK 88.0
END DESCRIPTION:
XS GIS Cut Line= 3
        2359025.     13770524.98        2358975.       13770325.
      2358475.01     13769125.04
#Sta/Elev= 30
    4785  515.18  4899.1  510.34  4908.7  510.07  4931.9   506.8  4949.9  500.39
  4970.8  490.41  4980.8  486.48  4988.6  480.75  4993.8  480.75  5000.3  475.39
  5015.1  474.43  5015.6  473.93  5032.1  474.43  5045.3  481.46  5053.4   483.9
  5082.7  484.13  5106.5  488.31  5121.1  488.92  5188.8  487.44  5229.5  489.99
  5520.3  492.43  5752.8  490.22  5879.5  492.65    5908  494.84  5992.7   502.3
  6016.5  505.75    6075  509.71  6128.6  516.13  6269.5  524.57  6291.1  527.01
#Mann= 7 ,-1 , 0
    4785     .07       0  4899.1     .12       0  4970.8      .1       0
  5015.1     .05       0  5032.1      .1       0  5752.8     .07       0
    5908     .12       0
Bank Sta=5015.1,5032.1
XS Rating Curve= 0 ,0
Exp/Cntr=0.3,0.1

Type RM Length L Ch R = 1 ,53553   ,312,312,312
BEGIN DESCRIPTION:
NASH CREEK 87.0
END DESCRIPTION:
XS GIS Cut Line= 3
        2359275.     13770425.01        2359275.       13770025.
      2358675.03     13769425.03
#Sta/Elev= 30
    4600  512.81  4638.6  512.92    4650  512.61    4660  511.12    4680  506.75
    4710  496.41    4730  488.14    4740  486.13  4806.5  483.52    4860  482.96
    4890  483.85    4940  483.61    4970  480.09    4989  475.62  4989.5  475.12
    5006  475.62  5014.2  475.83  5028.3  481.83  5035.4  483.27  5042.4  486.15
  5056.6  486.96  5183.9  487.43  5325.3  490.63  5523.3   490.3  5543.4  489.49
  5598.4  489.23  5707.1  490.11  5763.7  492.06    5792  493.65  5848.5  498.96
#Mann= 7 ,-1 , 0
    4600     .07       0  4638.6     .12       0  4806.5      .1       0
    4989     .05       0    5006      .1       0  5543.4     .12       0
  5598.4     .07       0
Bank Sta=4989,5006
XS Rating Curve= 0 ,0
Exp/Cntr=0.3,0.1

Type RM Length L Ch R = 1 ,53241   ,317,317,317
BEGIN DESCRIPTION:
B19768
END DESCRIPTION:
XS GIS Cut Line= 4
        2359435.     13770708.51      2359625.02     13769990.67
      2359403.34     13769684.53      2358739.17      13769104.7
#Sta/Elev= 30
  4066.9  513.47    4174  514.16  4316.8  508.19  4325.7  507.54  4347.4  506.61
  4420.1  503.29  4443.1  502.02  4513.2  492.21  4619.7  488.26  4736.8  486.81
  4814.4  486.24  4935.6  486.54  4950.3  485.67  4998.2  475.83  4998.7  475.33
  5015.2  475.83  5042.3  481.05  5063.4  478.59  5092.5  480.31  5100.4  482.48
  5142.8  484.06  5264.3  482.85    5312  485.59  5334.5  487.37  5434.2  487.98
  5672.1  494.12  5851.9   499.7  5931.5  507.16  6015.2  514.92  6069.1  516.19
#Mann= 13 ,-1 , 0
  4066.9     .12       0  4316.8     .07       0  4325.7     .12       0
  4347.4     .07       0  4420.1     .12       0  4619.7      .1       0
  4736.8     .12       0  4814.4      .1       0  4998.2     .05       0
  5015.2      .1       0    5312     .12       0  5672.1     .07       0
  5931.5     .12       0
Bank Sta=4998.2,5015.2
XS Rating Curve= 0 ,0
Exp/Cntr=0.3,0.1

Type RM Length L Ch R = 1 ,52924   ,260,260,260
BEGIN DESCRIPTION:
B19767
END DESCRIPTION:
XS GIS Cut Line= 4
      2359561.69     13770687.36      2359825.59     13769969.55
      2359688.36     13769515.63      2358855.72     13768999.18
#Sta/Elev= 30
  3872.1  512.58  3938.5  512.69  4002.5  511.06  4162.3  499.58  4330.9  493.85
  4390.1  492.47  4434.3  489.55  4501.3  487.38  4623.2  486.09  4712.5  483.77
  4831.9  485.89    4936  485.14    4969  484.03  4996.7  481.68  5009.2  474.83
  5009.7  474.33  5026.3  474.83  5034.9  475.66  5049.1  479.51  5059.5  480.51
  5231.2  482.09  5289.1  481.32  5310.4  481.79  5326.9  484.05    5347  488.73
  5374.1     491  5557.2  492.12  5747.9  496.09  5877.4  499.51  6090.9  508.61
#Mann= 8 ,-1 , 0
  3872.1     .12       0  4330.9     .07       0  4434.3     .12       0
  4712.5      .1       0  5009.2     .05       0  5026.3      .1       0
  5326.9     .12       0  5747.9     .07       0
Bank Sta=5009.2,5026.3
XS Rating Curve= 0 ,0
Exp/Cntr=0.3,0.1

Type RM Length L Ch R = 1 ,52664   ,564,564,564
BEGIN DESCRIPTION:
B19766
END DESCRIPTION:
XS GIS Cut Line= 3
      2360100.07     13770687.43      2359941.71     13769642.31
      2359941.71     13768533.86
#Sta/Elev= 30
  3825.6  508.05  3868.5  506.76  3979.8  498.65  4083.7  495.06  4227.1  489.06
  4393.9  486.75    4415  486.38  4546.2  486.17  4629.6   483.3  4667.5  479.51
  4701.8   481.8    4930  481.16    5001   477.7  5001.5   477.2    5019   477.7
    5020  479.22  5031.4  480.05    5080  480.19    5110  484.31    5195  485.52
    5400  484.95  5481.8  489.02    5550  499.93    5560  498.29    5670   498.5
    5730  505.65    5750  505.11  5825.6  511.01    5890  515.67  5991.1  518.68
#Mann= 11 ,-1 , 0
  3825.6     .07       0  4083.7     .12       0  4393.9     .07       0
    4415     .12       0  4701.8      .1       0    5001     .05       0
    5019      .1       0  5031.4    .035       0    5195     .07       0
  5481.8     .12       0  5825.6     .07       0
Bank Sta=5001,5019
XS Rating Curve= 0 ,0
Exp/Cntr=0.3,0.1

Type RM Length L Ch R = 1 ,52100   ,388,388,388
BEGIN DESCRIPTION:
B19765
END DESCRIPTION:
XS GIS Cut Line= 3
      2360195.07     13770592.37      2360311.19     13769367.84
      2360195.13     13768439.39
#Sta/Elev= 30
  4229.6  503.85  4337.5  501.12  4528.3   499.5  4588.6  495.87  4627.7  495.16
  4869.5  491.47  4935.2  488.13  4960.2  486.91  4990.4  478.16  5000.4  476.42
  5001.3   474.8  5001.8   474.3  5019.7   474.8  5030.5  476.79  5050.6  476.76
  5060.7   475.4  5100.9   478.9  5132.4  478.63    5231  479.49  5360.6  480.63
  5447.2  481.76  5634.6  488.15    5654  489.65  5744.2  490.81  5845.4  494.67
  5952.1  504.18  5996.6  509.51    6047  512.61    6194  517.02  6395.3  528.33
#Mann= 10 ,-1 , 0
  4229.6     .07       0  4627.7     .12       0  4869.5     .07       0
  4935.2     .12       0  5001.3     .05       0  5019.7     .12       0
  5132.4      .1       0    5231    .035       0  5360.6     .07       0
  5744.2    .035       0
Bank Sta=5001.3,5019.7
XS Rating Curve= 0 ,0
Exp/Cntr=0.3,0.1

Type RM Length L Ch R = 1 ,51712   ,388,388,388
BEGIN DESCRIPTION:
B19764
END DESCRIPTION:
XS GIS Cut Line= 3
      2360722.88     13770571.24      2360585.65     13769642.31
      2360290.07     13768523.31
#Sta/Elev= 30
  4338.9  509.74  4563.2  498.32  4810.2  493.94  4975.7     488  4992.2  483.51
  5002.3  476.93  5003.2  470.89  5003.7  470.39  5021.6  470.89  5032.6  472.49
  5040.3  476.01  5052.8  477.59  5140.8  478.44  5234.8  477.13  5317.8  477.69
  5442.7     481  5536.9  482.11  5577.2  483.63  5617.5  483.47  5637.1  484.88
  5962.1  492.66    6036  495.88  6061.2  497.98  6154.3  502.13  6222.6  508.16
  6247.4  511.28  6268.1  511.94  6288.7  511.07  6330.1  515.05  6435.3   521.3
#Mann= 9 ,-1 , 0
  4338.9     .07       0  5003.2     .05       0  5021.6     .07       0
  5140.8    .035       0  5317.8     .12       0  5442.7     .07       0
  5962.1    .035       0    6036     .07       0  6222.6    .035       0
Bank Sta=5003.2,5021.6
XS Rating Curve= 0 ,0
Exp/Cntr=0.3,0.1

Type RM Length L Ch R = 1 ,51324   ,408,408,408
BEGIN DESCRIPTION:
B19763
END DESCRIPTION:
XS GIS Cut Line= 4
      2361124.04     13770476.31      2360965.68     13769821.76
        2360744.     13769578.97      2360437.86     13768533.88
#Sta/Elev= 30
  4117.2  503.81  4190.6  502.66  4290.8   497.4  4427.1  493.76  4447.8   491.5
  4494.8  492.98  4604.7  493.04  4660.5  489.83    4705  484.93  4804.3  482.63
  4859.5  481.97  4880.1  475.22  4923.1  472.55  4941.2  475.16  4958.8  474.96
  4963.8  470.71  4964.3  470.21  4982.3  470.71  5001.4  474.41  5022.4  475.53
  5079.1   474.2  5100.1  474.83  5118.7  477.59  5191.7  478.38    5218  479.45
  5701.2  490.15  5812.4  493.29  6071.8  504.06  6123.9  507.28  6208.4  516.36
#Mann= 13 ,-1 , 0
  4117.2     .07       0  4290.8     .12       0  4494.8     .07       0
  4660.5    .035       0  4804.3     .12       0  4880.1    .035       0
  4941.2      .1       0  4963.8     .05       0  4982.3      .1       0
  5191.7     .12       0    5218     .07       0  5701.2    .035       0
  5812.4     .07       0
Bank Sta=4963.8,4982.3
XS Rating Curve= 0 ,0
Exp/Cntr=0.3,0.1

Type RM Length L Ch R = 1 ,50916   ,519,519,519
BEGIN DESCRIPTION:
B19762
END DESCRIPTION:
XS GIS Cut Line= 3
      2361335.15     13770243.99      2361071.24     13769167.27
      2360849.88     13768450.46
#Sta/Elev= 30
  4259.8  494.89  4282.6  494.62  4492.5  489.54  4594.6  487.36  4855.9  476.04
  4906.9  476.58  4958.9  472.82  4979.5  473.51  4991.1  467.93  4991.6  467.43
  5009.6  467.93    5031  472.76  5061.8  472.55  5083.6  475.65  5138.9   475.8
  5195.7  480.63  5403.5  484.53  5542.8  486.66  5619.9  489.67  5663.8  489.87
  5711.2  493.03  5716.4  492.04  5749.1  494.41  5781.7  494.09  5828.3  497.07
  5862.7  497.21  5894.1  500.17  5917.5  499.94  6030.1  504.83  6118.6  510.21
#Mann= 10 ,-1 , 0
  4259.8     .07       0  4282.6    .035       0  4492.5     .07       0
  4594.6     .12       0  4991.1     .05       0  5009.6     .12       0
  5138.9     .07       0  5403.5    .035       0  5619.9     .12       0
  5828.3     .07       0
Bank Sta=4991.1,5009.6
XS Rating Curve= 0 ,0
Exp/Cntr=0.3,0.1

Type RM Length L Ch R = 1 ,50397   ,455,455,455
BEGIN DESCRIPTION:
NASH CREEK 82.0
END DESCRIPTION:
XS GIS Cut Line= 3
        2361625.     13769924.98        2361575.       13769575.
      2361075.01     13768375.03
#Sta/Elev= 30
  4646.1  490.54  4706.7  485.79  4853.2  480.13  4878.4  479.43  4908.7  473.96
    4939  472.63  4959.2  470.59    4960  469.51  4960.5  469.01  4978.6  469.51
  5091.2   473.6  5205.5  473.99  5237.9  472.63  5421.9   479.1  5607.1  482.64
  5732.2  484.72  5844.2  488.15  5931.3  492.41  5948.1  494.62  5963.8  494.41
  5971.9  496.48    6018   499.6  6054.3  500.35  6078.1  503.87  6123.6  507.64
  6131.2   507.1    6155  510.64  6208.1  514.87  6261.2  517.19  6299.6  520.69
#Mann= 10 ,-1 , 0
  4646.1     .07       0  4853.2     .12       0    4960     .05       0
  4978.6     .12       0  5237.9     .07       0  5421.9    .035       0
  5607.1     .07       0  5732.2     .12       0  5844.2     .07       0
  6123.6     .12       0
Bank Sta=4960,4978.6
XS Rating Curve= 0 ,0
Exp/Cntr=0.3,0.1

Type RM Length L Ch R = 1 ,49942   ,447,447,447
BEGIN DESCRIPTION:
NASH CREEK 81.0
END DESCRIPTION:
XS GIS Cut Line= 3
        2361875.     13769824.97        2361925.       13769375.
      2361324.99     13768824.99
#Sta/Elev= 30
  4546.8  485.12  4647.4  483.52  4697.7  479.71  4777.3  476.36  4788.2  475.56
  4798.3  471.56  4818.4   470.2  4848.6  470.11  4868.7  471.64  4928.2  471.25
  4939.2  468.67  4949.2  468.24  4959.3  469.73    4997  465.45  4997.3  464.46
  4997.8  463.96  5015.9  464.46  5020.8  469.52    5031  469.96  5041.2   470.5
  5063.4  471.52  5084.3  476.08  5091.7  475.45  5112.7  478.09  5161.1  480.23
  5191.6  481.07  5565.9  480.96  5629.4   481.3  5650.1  482.55  5813.5  485.25
#Mann= 10 ,-1 , 0
  4546.8     .07       0  4777.3     .12       0  4928.2      .1       0
  4997.3     .05       0  5015.9      .1       0    5031     .12       0
  5041.2     .07       0  5161.1     .12       0  5191.6    .035       0
  5650.1     .07       0
Bank Sta=4997.3,5015.9
XS Rating Curve= 0 ,0
Exp/Cntr=0.3,0.1

Type RM Length L Ch R = 1 ,49495   ,468,468,468
BEGIN DESCRIPTION:
NASH CREEK 80.0
END DESCRIPTION:
XS GIS Cut Line= 3
      2362374.99     13769774.95        2362325.       13769325.
      2361425.01     13768125.02
#Sta/Elev= 30
  4547.6   483.7  4799.1  474.83  4929.9     473  4965.6  468.06  4980.2  466.94
  4988.5  461.82    4989  461.32  5007.1  461.82  5007.6  462.99  5013.9     463
  5022.2  468.38  5057.6  471.96  5082.2  472.43    5143  475.18  5203.9  475.74
  5207.9  475.79  5812.3  481.15  5916.6  484.97  5963.9  489.85  6050.3  505.41
  6107.6  512.46  6257.6  523.27  6272.2  523.79  6278.4  522.48  6286.8  524.27
    6293  522.68  6309.9  527.02  6313.9  526.33  6357.6  533.23  6500.3  541.26
#Mann= 10 ,-1 , 0
  4547.6     .07       0  4965.6      .1       0  4988.5     .05       0
  5007.1      .1       0  5082.2    .035       0  5203.9     .07       0
  5207.9    .035       0  5812.3     .07       0  5916.6     .12       0
  6309.9     .07       0
Bank Sta=4988.5,5007.1
XS Rating Curve= 0 ,0
Exp/Cntr=0.3,0.1

Type RM Length L Ch R = 1 ,49027   ,463,463,463
BEGIN DESCRIPTION:
NASH CREEK 79.0
END DESCRIPTION:
XS GIS Cut Line= 3
      2362825.01     13769625.04        2362775.       13769275.
      2361574.98     13768174.98
#Sta/Elev= 30
  4651.6  484.56  4712.3  483.14  4762.8  478.38  4904.2  472.52  4924.4  469.14
  4957.9  468.48    4985   464.5  4985.7  463.19  4986.2  462.69  5004.4  463.19
  5005.2     465  5012.3  463.51  5019.1  470.13  5026.5  468.51  5111.6  470.19
  5189.3  469.48  5203.4  471.48  5260.2  467.96  5316.9  474.67  5364.3  474.93
  5614.1  479.28  5981.9  479.98  6088.3  483.45  6171.6  489.87  6236.9  494.37
  6300.4  507.57  6413.9  519.74    6449  525.19  6546.2  532.29  6633.1  535.53
#Mann= 7 ,-1 , 0
  4651.6     .07       0  4957.9     .12       0  4985.7     .05       0
  5004.4     .12       0  5364.3     .07       0  6171.6     .12       0
  6546.2     .07       0
Bank Sta=4985.7,5004.4
XS Rating Curve= 0 ,0
Exp/Cntr=0.3,0.1

Type RM Length L Ch R = 1 ,48564   ,334,334,334
BEGIN DESCRIPTION:
NASH CREEK 78.0
END DESCRIPTION:
XS GIS Cut Line= 3
      2363225.01     13769425.03        2363175.       13769175.
      2361974.97     13768074.97
#Sta/Elev= 30
  4745.1  482.05  4949.1  475.41  4959.3  474.13    4977  467.98  4988.1  460.94
  4988.6  460.44  5006.9  460.94  5021.4  460.99  5035.5  462.99  5042.3  467.42
  5056.5  468.64  5261.8  470.76  5290.2  469.98  5304.4  467.31  5325.7   466.5
  5382.1  470.65  5403.7  470.77  5410.4  469.35  5467.2  472.81  5506.3  473.46
  6026.4  479.75  6125.7  484.84  6207.8  492.62  6281.1  497.51  6295.3  497.94
  6309.5  496.42  6401.4  507.32  6458.1  509.97  6495.8  514.63    6628  518.94
#Mann= 7 ,-1 , 0
  4745.1     .07       0    4977     .12       0  4988.1     .05       0
  5006.9     .12       0  5506.3     .05       0  6207.8     .12       0
  6495.8     .07       0
Bank Sta=4988.1,5006.9
XS Rating Curve= 0 ,0
Exp/Cntr=0.3,0.1

Type RM Length L Ch R = 1 ,48230   ,581,581,581
BEGIN DESCRIPTION:
B19761
END DESCRIPTION:
XS GIS Cut Line= 4
      2363604.77     13769705.63      2363499.21     13769114.49
       2363140.3     13768533.89       2362897.5     13767752.72
#Sta/Elev= 30
  4353.5  499.27  4383.5  496.32  4506.5  487.17  4608.2  483.03  4650.1  481.66
  4882.4  476.61  4933.2  473.52  4973.4  464.95  4980.9  463.83    4991   463.2
  4991.5   462.7  5009.9   463.2  5013.8   466.2  5023.3  467.12  5094.5  463.47
  5117.9  464.72  5123.8  467.26  5241.5  467.66  5376.7  465.57    5450  470.99
  5486.7  470.33    5502  468.01  5821.8  472.56  5883.3  474.16  5987.4  479.72
  6041.2  482.74  6110.6  487.44  6175.7  497.72  6385.2  501.89  6454.6  502.73
#Mann= 14 ,-1 , 0
  4353.5     .12       0  4383.5     .07       0  4608.2     .12       0
  4650.1     .07       0  4973.4     .12       0  4980.9      .1       0
    4991     .05       0  5009.9      .1       0  5241.5     .12       0
  5821.8     .05       0  5883.3     .12       0  5987.4     .07       0
  6041.2     .12       0  6385.2     .07       0
Bank Sta=4991,5009.9
XS Rating Curve= 0 ,0
Exp/Cntr=0.3,0.1

Type RM Length L Ch R = 1 ,47649   ,469,469,469
BEGIN DESCRIPTION:
B19760
END DESCRIPTION:
XS GIS Cut Line= 4
      2364090.35     13769505.03      2363657.56     13768681.67
      2363467.54     13768491.66      2363099.05     13767933.65
#Sta/Elev= 30
  3953.1  500.56  3980.4  499.27    4127  492.67  4171.8  488.51  4275.7  478.22
  4446.4     473  4625.9   470.8  4793.4  469.84  4831.9  467.17  4837.5  463.85
  4859.6  462.99    4911  464.74  4939.3  463.09  4988.8  463.56  5007.5  459.86
    5008  459.36  5026.6  459.86  5031.2  461.62  5066.6  465.29  5116.1  466.39
  5150.3  472.58    5256  474.38  5272.9  474.54  5369.3  474.77  5454.8  475.52
  5604.6   481.4  5614.6  481.88  5734.9  489.67  5775.7  491.88  5820.7  493.38
#Mann= 13 ,-1 , 0
  3953.1     .07       0  3980.4     .12       0  4171.8     .07       0
  4625.9     .12       0  5007.5     .05       0  5026.6     .12       0
    5256     .07       0  5272.9     .12       0  5369.3     .07       0
  5604.6     .05       0  5614.6     .07       0  5734.9     .05       0
  5775.7     .12       0
Bank Sta=5007.5,5026.6
XS Rating Curve= 0 ,0
Exp/Cntr=0.3,0.1

Type RM Length L Ch R = 1 ,47180   ,486,486,486
BEGIN DESCRIPTION:
NASH CREEK 76.0
END DESCRIPTION:
XS GIS Cut Line= 3
      2364124.99     13769424.97        2363825.       13768225.
      2363574.97     13767974.97
#Sta/Elev= 30
    3767  499.36  3818.5  497.11  3866.9  493.07  3913.9  487.76  3961.2  484.56
  3982.9  482.99  4055.6   476.2  4096.8  473.93  4197.3  471.31  4291.7  470.68
  4568.4  469.51  4632.8  468.24    4705  464.13  4746.2  466.46    4857  466.25
  4952.4  460.96  4962.7  459.83  4971.2  455.43  4971.7  454.93  4990.3  455.43
  4993.6  458.72  5001.3  462.63  5007.4  462.63    5018  468.85  5032.2  471.32
  5074.6  471.72  5102.9  469.48  5151.8  472.47    5280  474.92  5357.5  476.38
#Mann= 9 ,-1 , 0
    3767     .12       0  3866.9     .07       0  3961.2     .12       0
  3982.9     .07       0  4291.7     .12       0  4971.2     .05       0
  4990.3     .12       0  5151.8     .07       0    5280     .05       0
Bank Sta=4971.2,4990.3
XS Rating Curve= 0 ,0
Exp/Cntr=0.3,0.1

Type RM Length L Ch R = 1 ,46694   ,456,456,456
BEGIN DESCRIPTION:
NASH CREEK 75.0
END DESCRIPTION:
XS GIS Cut Line= 3
      2364875.02     13768825.02        2364275.       13768325.
      2363824.99     13767774.99
#Sta/Elev= 30
  4219.1  498.08  4232.8  496.86  4269.2   490.7  4290.1  489.54  4391.4  479.47
    4432  477.34  4724.2  469.09  4793.8  466.72    4816  463.66  4836.8  466.33
  4851.1  466.57  4879.7  463.26  4894.1   464.6  4900.6  467.23  4943.5  467.72
  4957.9  466.67  4978.7  461.44  4986.5  461.15    4993  454.84  5003.4  454.82
  5004.1  453.02  5004.6  452.52  5023.4  453.02  5028.2  453.57    5036  458.65
  5142.3  462.55  5219.8  467.23  5379.9  469.15  5681.9  473.52  5710.8   474.1
#Mann= 7 ,-1 , 0
  4219.1     .12       0  4391.4     .07       0  4724.2     .12       0
  5004.1     .05       0  5023.4     .12       0  5379.9     .07       0
  5681.9     .05       0
Bank Sta=5004.1,5023.4
XS Rating Curve= 0 ,0
Exp/Cntr=0.3,0.1

Type RM Length L Ch R = 1 ,46238   ,442,442,442
BEGIN DESCRIPTION:
NASH CREEK 74.0
END DESCRIPTION:
XS GIS Cut Line= 3
      2364974.98     13768524.97        2364675.       13768175.
      2363475.02     13767075.01
#Sta/Elev= 30
  4539.1  490.23  4574.7  489.16  4624.1  485.39  4702.1  474.47  4744.9  471.17
  4823.9  469.72  4921.6   468.2  4972.6  464.33    4987  454.82  4987.5  454.32
  5006.4  454.82  5028.1  459.59  5042.3  460.96  5092.2  458.38  5106.4  460.57
  5191.4   461.1  5365.9  463.92  5492.3  466.71  5626.2  469.63  5642.8  469.43
    5736  469.31  5863.6  471.83  5955.5  475.82  5988.5  478.71  6004.8  481.48
  6075.7  481.05  6211.7  485.63  6380.3  493.53  6478.8  499.88  6627.9   507.6
#Mann= 13 ,-1 , 0
  4539.1     .12       0  4823.9     .07       0  4972.6     .12       0
    4987     .05       0  5006.4     .12       0  5191.4     .05       0
  5365.9     .12       0  5492.3     .05       0  5626.2     .07       0
  5642.8     .05       0  5988.5     .12       0  6211.7     .05       0
  6478.8     .07       0
Bank Sta=4987,5006.4
XS Rating Curve= 0 ,0
Exp/Cntr=0.3,0.1

Type RM Length L Ch R = 1 ,45796   ,471,471,471
BEGIN DESCRIPTION:
NASH CREEK 73.0
END DESCRIPTION:
XS GIS Cut Line= 3
      2365324.98     13768224.98        2365025.       13767925.
      2363824.99     13766924.99
#Sta/Elev= 30
  4570.9   488.7  4606.2  486.22  4641.6  478.92    4684  474.29  4740.6  471.22
  4825.4  470.44  4853.7  462.48  4867.9  460.39  4896.1  462.31  4910.3  468.32
  4924.4  464.97  4991.6  456.49  5002.3  456.54  5006.9  454.05  5007.4  453.55
  5026.3  454.05  5030.9  457.25  5037.4  457.86  5059.6  456.36  5073.2  458.87
  5129.9  457.43  5184.5  461.18  5293.9  461.14  5357.7     464  5627.1  464.23
  5726.1  468.34  5858.7  473.05  6060.6  479.87    6373  487.48  6557.2  498.59
#Mann= 6 ,-1 , 0
  4570.9     .07       0  5006.9     .05       0  5026.3     .07       0
  5184.5     .05       0  5726.1     .07       0  5858.7     .05       0
Bank Sta=5006.9,5026.3
XS Rating Curve= 0 ,0
Exp/Cntr=0.3,0.1

Type RM Length L Ch R = 1 ,45325   ,439,439,439
BEGIN DESCRIPTION:
NASH CREEK 72.0
END DESCRIPTION:
XS GIS Cut Line= 3
        2365825.       13767825.        2365325.       13767575.
      2364425.01     13766675.01
#Sta/Elev= 30
    4441  495.13  4463.4  494.36  4552.8  482.25  4566.8   481.3  4589.1   484.4
  4605.9  478.96  4611.5  480.65  4617.9  478.33  4762.4  470.51  4807.2  466.59
  4821.1  463.25  4874.2  466.67  4924.6  466.13  4963.7  461.27  4997.2  452.08
  5004.5  452.01    5005  451.51  5023.9  452.01  5031.9  456.13  5042.4  458.77
  5141.2  457.69  5282.9   460.8  5523.3  460.59  5608.1  467.76    5891  473.24
    5990  479.53  6018.3  483.98  6041.2  484.07  6100.9   484.6  6272.8  491.55
#Mann= 8 ,-1 , 0
    4441     .07       0  4617.9    .035       0  5004.5    .035       0
  5023.9    .035       0  5031.9     .05       0  5141.2    .035       0
  6041.2     .07       0  6100.9    .035       0
Bank Sta=5004.5,5023.9
XS Rating Curve= 0 ,0
Exp/Cntr=0.3,0.1

Type RM Length L Ch R = 1 ,44886   ,482,482,482
BEGIN DESCRIPTION:
NASH CREEK 71.0
END DESCRIPTION:
XS GIS Cut Line= 3
      2365875.01     13767525.01        2365625.       13767275.
      2364425.01     13766575.01
#Sta/Elev= 30
  4642.6   479.5  4847.5  461.45  4925.5  458.88    4982  458.53  4994.3  451.12
  4994.8  450.62  5013.8  451.12  5041.2  456.62  5062.7  458.31  5135.1  457.42
  5158.2  458.76  5218.4  457.29  5287.7  456.29  5331.9   459.4  5436.1  460.64
    5501  464.05  5636.2  466.42  5690.8  467.53  5720.1   466.3  5757.4  467.59
  5778.9  466.83    5955  470.12  6099.7  478.17  6115.4  481.59  6121.2  481.21
  6136.9  483.48  6179.9  483.43  6217.1  485.58  6275.8  491.23  6385.4  492.77
#Mann= 6 ,-1 , 0
  4642.6    .035       0  4847.5     .07       0  4994.3     .05       0
  5013.8     .07       0  5218.4     .07       0  5636.2    .035       0
Bank Sta=4994.3,5013.8
XS Rating Curve= 0 ,0
Exp/Cntr=0.3,0.1

Type RM Length L Ch R = 1 ,44404   ,447,447,447
BEGIN DESCRIPTION:
NASH CREEK 70.0
END DESCRIPTION:
XS GIS Cut Line= 3
        2366125.       13767425.        2365525.       13766825.
      2364924.97     13766224.97
#Sta/Elev= 30
  4150.3  477.49  4185.7  477.31    4221  474.57  4327.1  471.27    4420   465.6
  4475.6  459.07    4518  457.49  4601.4  457.62  4638.3  458.42  4673.6  457.64
  4687.7  455.59  4701.8  456.22  4730.1  453.41  4786.7  455.96  4839.1  454.88
  4899.8   455.9  4984.7  452.99  5002.4  451.56  5003.2  450.14  5003.7  449.64
  5022.8  450.14  5027.1  452.36  5041.2  452.96  5069.5   461.7  5338.2  462.33
  5408.9  464.81  5507.9  464.85  5559.8  466.79  5722.9  468.69  5847.4  472.09
#Mann= 9 ,-1 , 0
  4150.3     .07       0    4420    .035       0  4601.4     .07       0
  4638.3     .12       0  4839.1     .07       0  5003.2     .05       0
  5022.8     .07       0  5559.8    .035       0  5722.9     .07       0
Bank Sta=5003.2,5022.8
XS Rating Curve= 0 ,0
Exp/Cntr=0.3,0.1

Type RM Length L Ch R = 1 ,43957   ,473,473,473
BEGIN DESCRIPTION:
NASH CREEK 69.0
END DESCRIPTION:
XS GIS Cut Line= 3
      2366425.01     13767025.01        2365825.       13766525.
        2364825.     13765324.99
#Sta/Elev= 30
  4223.7  480.05  4328.4  472.91  4473.1  463.34  4571.9  461.95    4650  455.94
  4862.2  456.29  4948.1   453.9  4973.4   448.9  4973.9   448.4  4993.1   448.9
    5008  449.64  5040.5  459.41  5054.9  457.44  5125.2  457.35  5196.7  458.22
  5211.1  461.09  5493.4  461.12  5565.1   461.7  5572.9  464.35  5579.4  462.24
  5587.3   464.7  5593.8  462.44  5601.6  464.78  5638.8  464.17  5835.9  466.16
  6197.8  476.26  6268.1  483.05  6374.8  486.18  6460.7   494.7  6566.8  499.09
#Mann= 7 ,-1 , 0
  4223.7     .07       0  4328.4    .035       0  4473.1     .07       0
  4973.4     .05       0  4993.1     .07       0  5493.4    .035       0
  5638.8     .07       0
Bank Sta=4973.4,4993.1
XS Rating Curve= 0 ,0
Exp/Cntr=0.3,0.1

Type RM Length L Ch R = 1 ,43484   ,448,448,448
BEGIN DESCRIPTION:
NASH CREEK 68.0
END DESCRIPTION:
XS GIS Cut Line= 3
      2366425.02     13766625.03        2366225.       13766325.
      2365024.98     13765224.98
#Sta/Elev= 30
  4635.3  466.52  4779.6     464  4859.2  458.96  4880.2  454.62  4917.4  457.38
  4931.3  457.96  4952.3   449.9  4978.5  446.83    4979  446.33  4998.3  446.83
  5023.9  451.05  5176.1  453.64  5392.1  455.77  5399.5  453.13  5406.2   456.1
  5731.8  458.01  5916.2  464.26  5951.3  462.96  5965.5  463.62  5979.7  469.85
  5986.5  467.06  5993.9  470.29  6000.7  467.82  6008.1  470.43  6014.9  468.09
  6142.5  471.79  6248.6  482.37  6404.6  486.69  6496.4  494.09  6623.8  495.71
#Mann= 5 ,-1 , 0
  4635.3     .07       0  4917.4     .12       0  4978.5     .05       0
  4998.3     .12       0  5176.1     .07       0
Bank Sta=4978.5,4998.3
XS Rating Curve= 0 ,0
Exp/Cntr=0.3,0.1

Type RM Length L Ch R = 1 ,43036   ,508,508,508
BEGIN DESCRIPTION:
NASH CREEK 67.0
END DESCRIPTION:
XS GIS Cut Line= 3
      2366724.99       13766175.        2366175.       13765925.
      2365275.01     13765325.01
#Sta/Elev= 30
  4395.7  464.79    4433  466.04  4450.6  463.78    4545  462.66  4617.2  461.84
  4799.8  459.95  4847.2  458.45  4887.8  452.12  4916.4  450.94  4933.9  445.18
  5007.4  446.36  5018.4  444.47  5018.9  443.97  5038.4  444.47  5043.4  449.33
  5049.4  445.27  5058.4  448.53  5064.4  446.54    5072  450.14  5121.9  451.56
  5144.1  454.41  5373.9     455  5671.4  461.32  5749.5  464.52  5857.7  477.95
  5901.2  481.13  5965.8  485.25  5980.9  484.03  6037.9  489.64  6081.5  488.63
#Mann= 7 ,-1 , 0
  4395.7    .035       0    4545     .07       0  4617.2    .035       0
  4799.8     .12       0  5018.4     .05       0  5038.4     .12       0
  5121.9     .07       0
Bank Sta=5018.4,5038.4
XS Rating Curve= 0 ,0
Exp/Cntr=0.3,0.1

Type RM Length L Ch R = 1 ,42528   ,568,568,568
BEGIN DESCRIPTION:
NASH CREEK 66.0
END DESCRIPTION:
XS GIS Cut Line= 3
      2366975.01     13766075.01        2366175.       13765475.
      2365374.95     13765324.99
#Sta/Elev= 30
  3999.9  474.83  4007.5  474.77  4057.2  474.28  4107.2  469.32    4178   466.3
    4228  461.46  4236.4   463.9  4242.6  461.96  4263.5  464.97  4271.8  462.78
  4307.2  461.27  4642.6  456.06  4692.6  450.65    4915  448.44  4999.9  444.79
  5000.1  443.53  5000.6  443.03  5020.1  443.53  5040.6   444.4    5061  450.23
  5083.8  451.75  5447.6  462.49  5514.6  463.14  5640.9   472.1  5661.2   468.5
  5671.4   475.4  5677.3  477.06  5682.4  476.38  5701.9   479.5  5813.9  489.41
#Mann= 5 ,-1 , 0
  3999.9     .07       0  4007.5    .035       0    4915     .07       0
  5000.1     .05       0  5020.1     .07       0
Bank Sta=5000.1,5020.1
XS Rating Curve= 0 ,0
Exp/Cntr=0.3,0.1

Type RM Length L Ch R = 1 ,41960   ,550,550,550
BEGIN DESCRIPTION:
NASH CREEK 65.0
END DESCRIPTION:
XS GIS Cut Line= 3
        2367275.       13765825.        2366475.       13765025.
        2365675.       13764625.
#Sta/Elev= 30
  3868.7   467.9  3879.4  467.73  3939.4  464.85  4236.4  457.73  4448.5  455.17
  4575.8  456.57  4802.1  447.08  4842.9  446.98  4957.6  447.84  4985.9  443.15
  4986.5  441.78    4987  441.28  5006.6  441.78  5008.5  443.36    5014  442.35
  5022.4  445.71  5030.8  447.12  5044.8  447.84  5089.5  446.43  5215.3  448.29
  5281.4  451.18  5349.5  454.18  5416.7  454.96  5550.7  456.52  5670.9  460.13
  5693.3  464.75  5774.3  468.78  5805.1  477.64  5849.8  485.05  5894.5  487.61
#Mann= 7 ,-1 , 0
  3868.7     .07       0  3879.4    .035       0  4842.9     .07       0
  4986.5     .05       0  5006.6     .07       0  5281.4    .035       0
  5416.7     .07       0
Bank Sta=4986.5,5006.6
XS Rating Curve= 0 ,0
Exp/Cntr=0.3,0.1

Type RM Length L Ch R = 1 ,41410   ,556,556,556
BEGIN DESCRIPTION:
NASH CREEK 64.0
END DESCRIPTION:
XS GIS Cut Line= 3
      2368275.03     13764975.01        2366725.       13764625.
      2365975.01       13764075.
#Sta/Elev= 30
  3410.2   520.6    3447  515.58  3580.4  502.62  3684.6  493.64  3843.7  481.78
  3871.6  477.57  3951.9  472.83  4026.8  465.88  4322.6  452.18  4527.7  447.85
  4756.5  447.53  4794.7  445.26  4804.5  441.64    4825  447.35  4883.6  446.68
  4888.7  439.91  4916.7  437.81  4917.2  437.31  4936.9  437.81  4985.5  439.97
  5056.7  441.56  5098.5  445.72  5188.1  444.32  5363.4  452.79  5585.5  456.82
  5722.1  467.84  5792.9     482  5830.1  482.79  5857.2  487.84  5929.3  489.16
#Mann= 13 ,-1 , 0
  3410.2     .12       0    3447     .07       0  3580.4    .035       0
  3684.6     .07       0  3951.9    .035       0  4756.5     .07       0
  4794.7     .12       0  4916.7     .05       0  4936.9     .12       0
  4985.5     .07       0  5188.1    .035       0  5363.4     .07       0
  5722.1    .035       0
Bank Sta=4916.7,4936.9
XS Rating Curve= 0 ,0
Exp/Cntr=0.3,0.1

Type RM Length L Ch R = 1 ,40854   ,602,602,602
BEGIN DESCRIPTION:
NASH CREEK 63.0
END DESCRIPTION:
XS GIS Cut Line= 3
      2367875.02     13764825.02        2367075.       13764325.
        2366075.       13764075.
#Sta/Elev= 30
    4056  482.86    4079  481.66    4158  471.92  4223.4  467.92  4374.4  457.48
  4425.7  455.95  4577.8  446.96  4860.8  443.07  4949.3  442.34  4999.4  437.72
  4999.5  436.79    5000  436.29  5019.9  436.79  5022.6  439.27    5051  447.12
  5105.1  447.63  5140.5  449.38  5146.3  448.26  5215.9  447.39  5293.8  448.75
  5348.2  449.34  5512.2  452.08  5604.6  451.94  5710.7  453.46  5793.1  457.73
  5865.3  467.51  5924.5  481.39  5951.6  481.86  6012.2  482.42  6030.2   484.8
#Mann= 10 ,-1 , 0
    4056     .07       0  4223.4    .035       0  4860.8     .12       0
  4999.5     .05       0  5019.9     .12       0  5140.5    .035       0
  5293.8     .07       0  5348.2    .035       0  5604.6     .07       0
  5951.6    .035       0
Bank Sta=4999.5,5019.9
XS Rating Curve= 0 ,0
Exp/Cntr=0.3,0.1

Type RM Length L Ch R = 1 ,40252   ,499,499,499
BEGIN DESCRIPTION:
B19759
END DESCRIPTION:
XS GIS Cut Line= 3
      2368217.89     13764522.45      2367510.64     13764110.76
      2366149.39     13764015.79
#Sta/Elev= 30
  4312.8  496.61  4468.3  485.26  4501.8  482.89  4554.8  475.17  4715.3  464.06
  4860.1  448.36  4977.6  444.41    4983  434.31  4983.5  433.81  5003.5  434.31
  5036.3  438.49  5187.8  440.98  5371.6  445.88  5515.7  445.95  5726.6  448.35
  5957.5  451.76  5968.8  455.39  5978.8  455.13    6004  447.95    6039  449.75
  6079.1  447.86  6099.1   451.7  6122.9   451.7  6209.4  452.27  6309.6  456.49
  6369.8  464.51  6399.9  472.42  6419.9  481.18  6486.9  481.84  6495.7  481.64
#Mann= 11 ,-1 , 0
  4312.8     .07       0  4468.3     .12       0    4983     .05       0
  5003.5     .12       0  5187.8    .035       0  5371.6     .07       0
  5515.7    .035       0  5726.6     .07       0  5957.5    .035       0
  6122.9     .07       0  6486.9    .035       0
Bank Sta=4983,5003.5
XS Rating Curve= 0 ,0
Exp/Cntr=0.3,0.1

Type RM Length L Ch R = 1 ,39753   ,567,567,567
BEGIN DESCRIPTION:
NASH CREEK 62.0
END DESCRIPTION:
XS GIS Cut Line= 3
      2368274.97     13763525.01        2367675.       13763725.
      2366074.98       13763925.
#Sta/Elev= 30
  4367.6   503.6  4409.7  500.13  4451.9   491.4  4631.1   470.6  4652.2  465.56
  4704.9  464.69  4757.6  459.18  4834.9  455.31  4936.8   446.7  4989.5  439.54
  5002.5  436.98  5010.1  432.71    5020  432.56  5020.5  432.06  5040.5  432.56
  5042.9  436.39  5050.4  437.18  5119.1  439.04  5302.4  446.01  5440.9  443.77
    5558  447.57  5744.1  447.54  5953.7  448.85  6259.8  453.21  6350.5  456.84
  6413.4  465.54  6451.2  472.67  6481.5  480.77  6574.7  483.72  6612.5  487.56
#Mann= 9 ,-1 , 0
  4367.6     .07       0  4834.9     .12       0    5020     .05       0
  5040.5     .12       0  5119.1     .07       0    5558    .035       0
  5744.1     .07       0  5953.7    .035       0  6259.8     .07       0
Bank Sta=5020,5040.5
XS Rating Curve= 0 ,0
Exp/Cntr=0.3,0.1

Type RM Length L Ch R = 1 ,39186   ,370,370,370
BEGIN DESCRIPTION:
NASH CREEK 61.0
END DESCRIPTION:
XS GIS Cut Line= 3
      2368024.98     13763324.99        2367575.       13763225.
      2365975.04     13763874.98
#Sta/Elev= 30
  4533.2  477.65  4584.4   474.8  4615.1  465.14  4666.3  459.21  4698.4  458.96
  4723.8  465.25  4741.9  465.98  4758.5  454.58  4768.8  452.59  4963.4  441.01
  5005.4  431.22  5005.9  430.72    5026  431.22  5038.1  434.29  5069.7  438.87
  5155.1  439.04  5402.6  436.77  5431.9  442.28    5523  448.96  5624.3  448.93
    5879  448.15  6226.6  453.34  6321.8  459.17  6375.7  458.75  6392.4  461.96
  6414.6  467.69  6468.1  474.21  6559.2  484.17  6624.4  487.68  6721.1  488.13
#Mann= 11 ,-1 , 0
  4533.2     .07       0  4723.8     .12       0  5005.4     .05       0
    5026     .12       0  5038.1     .07       0  5155.1     .12       0
  5402.6    .035       0  5624.3     .07       0  6226.6    .035       0
  6392.4     .07       0  6624.4    .035       0
Bank Sta=5005.4,5026
XS Rating Curve= 0 ,0
Exp/Cntr=0.3,0.1

Type RM Length L Ch R = 1 ,38816   ,658,658,658
BEGIN DESCRIPTION:
B19758
END DESCRIPTION:
XS GIS Cut Line= 4
      2368312.95     13762928.45      2367531.75     13762854.55
      2367236.17     13763044.57      2366191.08     13763160.69
#Sta/Elev= 30
  4015.7  475.78  4190.4  467.12  4686.6  445.03  4908.9  439.75  4949.4  439.65
  4963.7   437.2  4968.5   429.3    4969   428.8  4989.1   429.3  5051.5  437.91
  5154.9  437.63  5201.6  434.77  5250.5  441.34  5424.6  442.37  5476.3  445.53
    5495  443.61  5652.4  445.51  5666.1  446.13  5684.7  452.16  5726.5  452.78
  5736.5  451.41    5748  443.96    5768  445.42  5829.3  448.52  5937.8  450.37
  5988.1  453.02  6002.2  456.44  6014.6   460.6  6068.6  466.94  6203.3   474.8
#Mann= 12 ,-1 , 0
  4015.7     .07       0  4190.4     .05       0  4908.9     .12       0
  4949.4     .07       0  4968.5     .05       0  4989.1     .07       0
  5201.6     .12       0  5250.5     .07       0  5684.7     .12       0
    5768     .07       0  5829.3     .12       0  6002.2     .07       0
Bank Sta=4968.5,4989.1
XS Rating Curve= 0 ,0
Exp/Cntr=0.3,0.1

Type RM Length L Ch R = 1 ,38158   ,657,657,657
BEGIN DESCRIPTION:
NASH CREEK 60.0
END DESCRIPTION:
XS GIS Cut Line= 3
      2368365.73     13762727.88      2367172.83     13762569.53
      2366339.46     13762495.69
#Sta/Elev= 30
  3618.7  478.43  3659.8  476.85  3676.8  473.96  3750.1  468.96    3800  467.06
  3906.8  462.68  3992.7  457.23  4105.4  453.75  4158.6  452.62  4440.1  444.98
  4476.9  443.11  4513.4  439.01  4591.7  436.31  4698.8  437.89  4740.9  436.75
  4789.6  434.26    4860  433.06  4950.4  434.11  4960.4  433.52  4970.2  429.43
  4970.7  428.93  4990.9  429.43  5030.7  436.76  5043.3  436.86    5280  442.52
  5422.2  452.83  5502.5  464.29  5552.7  468.99  5592.9  471.72  5658.7  472.77
#Mann= 9 ,-1 , 0
  3618.7     .07       0    3800     .05       0  4105.4    .035       0
  4158.6     .05       0  4740.9     .07       0  4970.2     .05       0
  4990.9     .07       0  5043.3    .035       0    5280     .07       0
Bank Sta=4970.2,4990.9
XS Rating Curve= 0 ,0
Exp/Cntr=0.3,0.1

Type RM Length L Ch R = 1 ,37501   ,584,584,584
BEGIN DESCRIPTION:
NASH CREEK 59.0
END DESCRIPTION:
XS GIS Cut Line= 3
      2368074.97     13762324.99        2367425.       13762175.
      2366275.01       13762375.
#Sta/Elev= 30
  4333.4  458.82  4384.7  456.96  4442.8  450.79  4456.5  452.48    4477  450.11
  4507.8  448.71  4836.2  443.92  4896.5  439.79  4918.3   438.7  4969.7  439.48
  4981.6  436.82  4987.5  426.86    4988  426.36  5008.3  426.86  5020.7  428.19
  5027.7  430.31    5065  431.52  5213.6  437.68  5391.2  436.99    5579  436.13
  5710.1  438.71  5771.9  440.02  5922.2  447.65    5985  459.58  6021.2  470.17
  6026.2  470.15  6035.8  474.14  6056.1  473.03  6127.1  478.87  6167.7   479.9
#Mann= 8 ,-1 , 0
  4333.4     .05       0  4896.5     .07       0  4987.5     .05       0
  5008.3     .07       0    5065    .035       0  5391.2     .05       0
  5710.1    .035       0  5922.2     .07       0
Bank Sta=4987.5,5008.3
XS Rating Curve= 0 ,0
Exp/Cntr=0.3,0.1

Type RM Length L Ch R = 1 ,36917   ,522,522,522
BEGIN DESCRIPTION:
NASH CREEK 58.0
END DESCRIPTION:
XS GIS Cut Line= 3
      2368125.04     13761975.02        2367325.       13761625.
      2366524.98     13761274.99
#Sta/Elev= 30
  4127.5  453.85  4293.2  447.76  4765.8  440.36  4835.1  440.38  4863.9  439.02
  4924.4  436.99  4957.1  434.03  4962.9  430.77  4968.4  431.89  4978.9  429.37
  4986.3  426.34  4987.6  424.57  4988.1  424.07  5008.4  424.57  5009.7  427.13
  5015.2  425.51  5022.6  428.59  5067.4  429.42  5114.2  433.77  5189.8  431.81
  5288.8  433.65    5513   432.8  5622.9  433.39  5655.7   430.7  5677.5  433.29
  5721.2  432.31  5737.1  434.38  5772.7  444.88  5812.8  457.05    5874   463.8
#Mann= 7 ,-1 , 0
  4127.5     .05       0  4765.8     .07       0  4863.9    .035       0
  4987.6    .035       0  5008.4    .035       0    5513      .1       0
  5772.7     .12       0
Bank Sta=4987.6,5008.4
XS Rating Curve= 0 ,0
Exp/Cntr=0.3,0.1

Type RM Length L Ch R = 1 ,36395   ,573,573,573
BEGIN DESCRIPTION:
NASH CREEK 57.0
END DESCRIPTION:
XS GIS Cut Line= 3
      2368675.03     13762275.02        2367125.       13761175.
      2366674.97     13761074.99
#Sta/Elev= 30
  3099.2  497.43    3132   495.5  3522.1   462.4  3704.4  454.74  3874.1  447.77
  3932.1  447.37  3945.3  450.09  3957.6  447.57  4363.7  440.81  4450.3  440.08
  4511.5  436.39  4608.1  435.85  4870.7  433.42  4900.3  428.89  4977.7  427.65
  4986.4  423.66  4986.9  423.16  5007.2  423.66  5030.6   428.7  5092.1  430.75
  5133.1  429.56    5160  425.07  5184.3  430.51  5226.8   433.5  5252.2  439.11
  5257.3  444.71  5262.7  446.59  5307.2  454.93  5442.6  465.23  5460.9  466.49
#Mann= 14 ,-1 , 0
  3099.2     .05       0    3132     .07       0  3522.1    .035       0
  3704.4     .05       0  3874.1     .07       0  3957.6     .05       0
  4363.7     .07       0  4450.3    .035       0  4608.1     .12       0
  4986.4     .05       0  5007.2     .12       0  5226.8      .1       0
  5262.7    .035       0  5442.6     .07       0
Bank Sta=4986.4,5007.2
XS Rating Curve= 0 ,0
Exp/Cntr=0.3,0.1

Type RM Length L Ch R = 1 ,35822   ,517,517,517
BEGIN DESCRIPTION:
NASH CREEK 56.0
END DESCRIPTION:
XS GIS Cut Line= 3
        2368275.       13761475.        2367475.       13760825.
      2366874.98     13760024.98
#Sta/Elev= 30
  3974.3  460.49    4095  449.11  4379.4  440.77  4393.8  435.36  4397.2  435.85
  4408.2  433.58  4414.6  435.51  4422.5  433.13    4429  434.68  4436.9  432.81
  4472.1  433.06  4486.5  433.69  4507.3  439.79  4515.2  439.26  4528.3  433.05
  4571.2  430.98  4663.9  433.02  4713.4  430.34  4834.8  430.96  4977.1  425.27
  4990.5  421.42    4991  420.92  5013.3  421.42  5026.9  432.43    5159  431.69
  5468.6  433.01  5518.6  435.98  5597.8  441.32  5733.8  445.35  6005.1  457.09
#Mann= 7 ,-1 , 0
  3974.3     .07       0  4397.2     .12       0  4990.5     .05       0
  5013.3     .12       0    5159     .07       0  5518.6     .12       0
  5733.8     .07       0
Bank Sta=4990.5,5013.3
XS Rating Curve= 0 ,0
Exp/Cntr=0.3,0.1

Type RM Length L Ch R = 1 ,35305   ,527,527,527
BEGIN DESCRIPTION:
NASH CREEK 55.0
END DESCRIPTION:
XS GIS Cut Line= 3
      2368524.98     13761424.97        2367925.       13760625.
        2367475.       13760075.
#Sta/Elev= 30
  4004.3  465.03  4226.1  449.67    4397  442.64  4411.6  440.74  4432.4  441.19
  4454.3  439.46  4461.6  440.42  4467.8  439.22  4538.7  438.13  4626.1  432.22
  4632.4  430.35  4661.6  427.29  4829.5  428.01  4867.8  426.29    4897  427.23
  4917.8  426.38  4938.5   422.6  4954.3  422.05  4964.7  419.25  4965.2  418.75
  4987.5  419.25  4990.7  428.27  5001.1  430.42  5023.3  430.79  5124.9  430.14
  5200.6   432.8    5366   435.7  5517.4  439.99  5583.8  441.42  5714.9  444.73
#Mann= 10 ,-1 , 0
  4004.3     .07       0  4538.7     .12       0  4829.5     .07       0
  4938.5     .12       0  4964.7     .05       0  4987.5     .12       0
  5023.3     .07       0  5200.6     .05       0  5517.4     .07       0
  5583.8     .05       0
Bank Sta=4964.7,4987.5
XS Rating Curve= 0 ,0
Exp/Cntr=0.3,0.1

Type RM Length L Ch R = 1 ,34778   ,547,547,547
BEGIN DESCRIPTION:
NASH CREEK 54.0
END DESCRIPTION:
XS GIS Cut Line= 3
      2368725.01     13760825.01        2368425.       13760525.
      2367624.97     13759774.97
#Sta/Elev= 30
  4571.1  442.75  4578.7   442.7  4660.2  440.48  4797.4  437.13  4810.2  433.95
  4825.7  426.88  4839.8  423.04    4854  423.34  4868.1  425.85  4967.1  424.86
  4991.8   418.5  4997.9  418.47  4998.4  417.97  5020.7  418.47  5023.5  421.13
  5030.8  421.92  5037.6  427.28    5045  427.31  5051.8  429.69  5129.9  431.05
  5207.6  430.49  5271.1  427.61  5346.6  429.11  5355.3  429.44  5639.4  432.49
  5773.7  437.75  5808.9  437.88  5879.7  440.79  5914.9  441.14    6092  448.32
#Mann= 8 ,-1 , 0
  4571.1     .07       0  4578.7     .12       0  4660.2     .07       0
  4810.2     .12       0  4997.9     .05       0  5020.7     .12       0
  5346.6     .07       0  5355.3     .05       0
Bank Sta=4997.9,5020.7
XS Rating Curve= 0 ,0
Exp/Cntr=0.3,0.1

Type RM Length L Ch R = 1 ,34231   ,544,544,544
BEGIN DESCRIPTION:
NASH CREEK 53.0
END DESCRIPTION:
XS GIS Cut Line= 3
        2369075.       13761025.        2368775.       13760225.
      2367974.98     13759424.98
#Sta/Elev= 30
  4145.5  463.81  4169.3  461.58  4209.6  458.64  4252.3  450.72  4287.3  448.27
  4393.6  444.13  4560.9  439.26  4673.3  436.82  4728.5  438.59  4783.6  438.31
  4899.3  433.99  4904.7  431.73  4924.3  429.16  4935.8  422.15  4946.5  418.96
  4948.4  415.25  4948.9  414.75  4971.3  415.25  5003.4  417.67  5028.2  423.69
  5056.5  426.37    5113  424.23  5141.3  427.29  5175.9   426.6  5268.6  425.47
  5381.7  428.64  5537.3  428.02  5795.3  429.92    6004   434.5  6131.3  442.17
#Mann= 9 ,-1 , 0
  4145.5     .07       0  4169.3    .035       0  4287.3     .07       0
  4393.6     .12       0  4560.9     .07       0  4948.4     .05       0
  4971.3     .07       0  5175.9     .05       0  5795.3     .07       0
Bank Sta=4948.4,4971.3
XS Rating Curve= 0 ,0
Exp/Cntr=0.3,0.1

Type RM Length L Ch R = 1 ,33687   ,553,553,553
BEGIN DESCRIPTION:
NASH CREEK 52.0
END DESCRIPTION:
XS GIS Cut Line= 3
      2369775.02     13760475.02        2369025.       13759775.
      2368325.02     13758625.03
#Sta/Elev= 30
  3974.5  459.83  4024.8  457.57  4278.6  444.13  4406.1  436.36  4505.3  435.55
  4526.3  429.71  4618.2  426.72  4731.5  429.03  4850.9  425.59  4887.3  423.53
  4897.4  427.02  4908.4  426.49  4915.7  420.12  4922.5  419.27  4936.7  424.66
    4965  424.35  4972.4  420.89  4974.8  415.24  4975.3  414.74  4998.2  415.24
  5040.7  420.03  5145.7  425.03  5237.4  424.97  5966.7  431.44  6042.4  434.15
  6143.3  445.74  6222.8  464.96  6262.3  469.74  6335.8  482.47  6346.7  483.73
#Mann= 12 ,-1 , 0
  3974.5     .12       0  4024.8     .07       0  4278.6     .12       0
  4850.9     .07       0  4897.4     .12       0  4974.8     .05       0
  4998.2     .12       0  5040.7     .07       0  5237.4     .05       0
  5966.7     .07       0  6262.3     .12       0  6335.8     .07       0
Bank Sta=4974.8,4998.2
XS Rating Curve= 0 ,0
Exp/Cntr=0.3,0.1

Type RM Length L Ch R = 1 ,33134   ,568,568,568
BEGIN DESCRIPTION:
NASH CREEK 51.0
END DESCRIPTION:
XS GIS Cut Line= 3
      2369925.02     13760075.02        2369175.       13759275.
      2368375.02     13758575.02
#Sta/Elev= 30
  3903.9  447.64  4123.2  436.46  4230.3  433.25  4625.6  428.07  4701.3  428.89
  4738.9  427.43  4781.2  422.48  4830.8  423.39  4873.3  420.78  4965.1  423.53
  4989.7  421.83  4997.1  418.87  5003.8  418.87  5007.6  415.78  5024.4  414.38
  5024.9  413.88  5047.8  414.38  5050.3  422.63  5066.2  425.96  5112.6  424.51
  5241.1  423.18  5691.4   429.6  5744.6  431.79  5808.7  439.19  5829.6  438.27
  5850.9  442.77  5909.8  450.07    5971   463.9  6021.3     479  6063.5  484.08
#Mann= 10 ,-1 , 0
  3903.9     .07       0  4230.3     .05       0  4701.3     .07       0
  4989.7     .05       0  5024.4     .05       0  5047.8     .05       0
  5066.2     .07       0  5112.6     .05       0  5691.4     .07       0
  5909.8     .12       0
Bank Sta=5024.4,5047.8
XS Rating Curve= 0 ,0
Exp/Cntr=0.3,0.1
