HEC-RAS study PEACH CREEK.prj: PEACH CREEK Base Level Engineering

--- PEACH CREEK.g01 (geometry) --- (continued)

Type RM Length L Ch R = 1 ,262674  ,965,965,965
BEGIN DESCRIPTION:
PEACH CREEK9145
END DESCRIPTION:
XS GIS Cut Line= 3
        2519575.     13853524.98        2519675.       13852575.
      2518824.97     13851274.96
#Sta/Elev= 30
  4044.4  410.69  4265.6  407.48  4305.8  408.06    4520  399.94  4771.4  394.03
  4818.6  394.07  4929.2  398.68  4953.1  395.57  4969.5  390.41    4976   385.1
  4976.5   384.6  5003.2   385.1  5007.2  397.12  5013.2  395.49  5028.3  398.86
  5049.4  399.45  5058.5  398.07  5094.7  397.62  5136.9  398.44  5188.2  395.92
  5281.6  398.44  5340.8  397.14    5382  398.87  5468.6  397.81  5640.8  400.96
  5700.1  402.03  5819.8  404.57  6333.3  408.74  6443.3  409.69  6552.9  410.92
#Mann= 11 ,-1 , 0
  4044.4     .12       0    4520     .05       0  4771.4      .1       0
    4976     .05       0  5003.2      .1       0  5340.8     .07       0
  5640.8     .12       0  5700.1     .07       0  5819.8     .05       0
  6333.3    .035       0  6443.3     .05       0
Bank Sta=4976,5003.2
XS Rating Curve= 0 ,0
Exp/Cntr=0.3,0.1

Type RM Length L Ch R = 1 ,261709  ,714,714,714
BEGIN DESCRIPTION:
PEACH CREEK9144
END DESCRIPTION:
XS GIS Cut Line= 3
      2521567.08     13854013.46      2520453.38     13852615.21
      2519424.98     13851174.97
#Sta/Elev= 30
  3163.4  406.95  3427.5  405.74    3669  397.98  3709.6  397.25  3797.6  395.99
  3888.8  395.35  4039.3   392.8  4312.3  396.79  4473.3  397.77  4569.6  395.13
  4626.1  392.89  4689.2  391.71  4758.4  393.94  4953.9  393.39  5000.4  385.98
  5001.9  381.68  5002.9  381.18  5042.5  381.68  5043.1  384.72  5078.8  393.32
  5108.2  392.98  5129.1  395.39  5143.9  392.65  5265.6  391.73  5441.8  394.41
  5572.2  395.23  5582.7  395.19  6315.4  401.74  6408.6  402.68  6720.7  407.02
#Mann= 17 ,-1 , 0
  3163.4     .12       0    3669     .07       0  3709.6     .12       0
  3797.6    .035       0  3888.8     .05       0  4312.3     .07       0
  4473.3     .05       0  4569.6     .07       0  4626.1     .05       0
  4689.2      .1       0  5001.9     .05       0  5042.5      .1       0
  5441.8     .05       0  5572.2    .035       0  5582.7     .05       0
  6315.4     .07       0  6408.6     .05       0
Bank Sta=5001.9,5042.5
XS Rating Curve= 0 ,0
Exp/Cntr=0.3,0.1

Type RM Length L Ch R = 1 ,260995  ,569,569,569
BEGIN DESCRIPTION:
PEACH CREEK9143
END DESCRIPTION:
XS GIS Cut Line= 3
      2521524.99     13853274.98        2521025.       13852575.
      2519424.99     13851124.99
#Sta/Elev= 30
  4135.7  406.87  4360.6  397.22  4493.3  393.53  4682.9  391.75  4810.3  392.06
  4896.4  388.57  4946.8  393.29  4999.3  391.64    5003  388.15  5003.6  380.34
  5004.6  379.84  5044.3  380.34  5045.6   386.9  5052.3  386.62  5059.8  390.06
  5066.5  389.52    5074  392.73  5300.4  391.94  5382.3  396.14  5477.4  400.04
  5600.5   400.5  5730.2  399.75    5822  399.76  6171.8  397.91  6619.4  401.74
  6836.5  403.45  6858.2  406.49  6942.6   404.4    7087  406.46  7155.2  407.19
#Mann= 12 ,-1 , 0
  4135.7     .07       0  4360.6     .05       0  4682.9      .1       0
  5003.6     .05       0  5044.3      .1       0  5382.3    .035       0
  5600.5     .05       0  5730.2    .035       0    5822     .12       0
  6171.8    .035       0  6619.4     .05       0    7087    .035       0
Bank Sta=5003.6,5044.3
XS Rating Curve= 0 ,0
Exp/Cntr=0.3,0.1

Type RM Length L Ch R = 1 ,260426  ,553,553,553
BEGIN DESCRIPTION:
PEACH CREEK9142
END DESCRIPTION:
XS GIS Cut Line= 3
      2522225.02     13853475.03        2521125.       13852075.
      2519524.98     13850624.98
#Sta/Elev= 30
  3214.8  411.44    3268  411.16  3371.2  411.96  3690.5  406.32  3735.1  405.51
    3826  404.19  4118.6  403.92  4211.1  401.51    4340  398.77  4736.2  394.56
  4917.5   389.5  4959.2  392.78  5023.3  387.77  5080.1  394.45  5249.8  390.18
    5251   387.5    5252     387  5291.7   387.5  5292.3  390.58  5370.7   392.8
  5554.5  393.16  5694.3   397.3  5752.6  400.15  5993.8  397.72  6530.7  401.38
  6784.9  404.86  6909.4  407.28  7042.3   408.9  7130.8   410.8  7154.6  411.11
#Mann= 17 ,-1 , 0
  3214.8     .12       0    3268     .07       0  3690.5     .05       0
  3735.1     .07       0    3826     .05       0  4211.1     .07       0
    4340     .05       0  4736.2      .1       0  5249.8     .05       0
    5251     .05       0  5291.7     .05       0  5694.3     .12       0
  6530.7     .05       0  6784.9    .035       0  6909.4     .05       0
  7042.3    .035       0  7130.8     .05       0
Bank Sta=5251,5291.7
XS Rating Curve= 0 ,0
Exp/Cntr=0.3,0.1

Type RM Length L Ch R = 1 ,259873  ,541,541,541
BEGIN DESCRIPTION:
PEACH CREEK9141
END DESCRIPTION:
XS GIS Cut Line= 3
      2522175.02     13852725.02        2521225.       13851625.
      2519624.97     13850624.98
#Sta/Elev= 30
  3546.6  404.13  3726.6  402.04  3929.8  402.63  4333.7  396.54  4819.8  396.71
  4879.9  395.93  4900.8  390.08  4915.1  393.26  4921.7  389.32  4929.3  391.32
  4950.2  385.14  4957.8  386.82  4964.4  382.91  4972.1  386.22  4978.7  383.02
  4986.3  385.29  4993.3  378.69  4994.3  378.19    5034  378.69  5035.5  383.36
    5059  391.65  5080.9  389.29  5499.6  391.22  5520.9  391.47  5741.2  397.63
  6312.2  400.04  6478.5  402.39  6651.7  404.59  6678.1  404.97  6886.9  410.06
#Mann= 11 ,-1 , 0
  3546.6     .07       0  3726.6     .05       0  4819.8      .1       0
  4993.3     .05       0    5034      .1       0  5499.6     .05       0
  5520.9     .12       0  6312.2    .035       0  6478.5     .05       0
  6651.7    .035       0  6678.1     .05       0
Bank Sta=4993.3,5034
XS Rating Curve= 0 ,0
Exp/Cntr=0.3,0.1

Type RM Length L Ch R = 1 ,259332  ,548,548,548
BEGIN DESCRIPTION:
PEACH CREEK9140
END DESCRIPTION:
XS GIS Cut Line= 5
      2524336.13       13851754.      2521115.37     13851203.26
        2521075.       13851175.      2521035.52     13851131.44
      2519162.46     13850142.86
#Sta/Elev= 30
  1683.1  424.31  1762.7  422.86    2605  403.25  2751.9  401.84  2873.5  401.71
  2986.2  401.38  3257.2  400.23  3676.2  390.98    3693  387.12  3775.7  389.57
  4008.7  389.46  4829.3  390.93  4977.6  391.26    5007  385.08  5007.6  378.69
  5008.6  378.19  5048.3  378.69  5049.6  386.65  5055.3  389.47  5160.9  389.56
  5552.8  398.49  5839.5  392.63  5943.5  399.58  6124.7  401.55  6218.8   403.3
  6415.2  407.61  6634.7  412.95  7015.2  422.84  7150.2  426.93  7176.6  427.21
#Mann= 20 ,-1 , 0
  1683.1    .035       0  1762.7     .05       0    2605    .035       0
  2751.9    .035       0  2873.5     .05       0  2986.2    .035       0
  3257.2     .07       0  3676.2     .12       0  3775.7      .1       0
  4008.7     .05       0  4829.3      .1       0  5007.6     .05       0
  5048.3      .1       0  5160.9     .12       0  6124.7     .12       0
  6218.8    .035       0  6415.2     .12       0  6634.7    .035       0
  7015.2     .12       0  7150.2     .07       0
Bank Sta=5007.6,5048.3
XS Rating Curve= 0 ,0
Exp/Cntr=0.3,0.1

Type RM Length L Ch R = 1 ,258784  ,581,581,581
BEGIN DESCRIPTION:
PEACH CREEK9139
END DESCRIPTION:
XS GIS Cut Line= 4
      2523843.05     13851073.44      2521625.83     13850842.01
        2521225.       13850675.      2520724.98     13850224.98
#Sta/Elev= 30
  2336.6  410.26  2621.7  404.45  2666.6  403.57  2913.1  401.79  3541.2  397.62
  3681.9   392.4  4136.9  388.09  4214.8  388.02  4285.2  385.31  4305.3  387.56
  4367.9  388.37  4415.9  390.13  4490.1  387.84  4624.7  390.78  4807.8   389.2
  4909.5  390.49  4990.9  390.06  5000.1  386.24    5001  378.26    5002  377.76
  5041.8  378.26  5049.8  385.11  5056.5  383.67  5078.2  386.61  5141.7  389.16
  5247.9  386.76  5269.2  389.89  5339.8  388.98  5375.6  390.86  5672.8  403.87
#Mann= 10 ,-1 , 0
  2336.6     .05       0  2621.7     .07       0  2666.6     .05       0
  2913.1    .035       0  4136.9      .1       0  4367.9     .05       0
  4909.5      .1       0    5001     .05       0  5041.8      .1       0
  5375.6     .05       0
Bank Sta=5001,5041.8
XS Rating Curve= 0 ,0
Exp/Cntr=0.3,0.1

Type RM Length L Ch R = 1 ,258203  ,563,563,563
BEGIN DESCRIPTION:
PEACH CREEK9138
END DESCRIPTION:
XS GIS Cut Line= 4
      2523481.98     13850649.83      2521477.08     13850213.72
        2521325.       13850125.      2519725.01     13849275.01
#Sta/Elev= 30
  2772.1     403  3229.5  397.46  3437.6  398.95  3577.5  399.52    3851  392.46
  4316.4  386.33  4414.7  383.48  4488.3  388.86  4496.2   383.7  4497.2   383.2
  4537.1   383.7  4539.5  389.26  4545.2  389.26  4927.9  389.71  4976.8   390.5
  5008.1  385.45  5079.7   390.1  5138.2  387.85  5288.2  390.28  5392.4  396.85
  5539.3  400.49  5590.3  400.97  5628.6  405.84  5672.5  400.32    5740  401.17
  5985.1  406.49  6185.4     414    6253  418.13  6673.6  436.81  6811.7  444.44
#Mann= 13 ,-1 , 0
  2772.1     .05       0  3437.6    .045       0  4316.4      .1       0
  4496.2     .05       0  4537.1      .1       0  4545.2     .05       0
  4927.9      .1       0  5138.2     .05       0  5539.3    .035       0
    5740     .05       0  6185.4     .07       0    6253     .05       0
  6673.6     .07       0
Bank Sta=4496.2,4537.1
XS Rating Curve= 0 ,0
Exp/Cntr=0.3,0.1

Type RM Length L Ch R = 1 ,257640  ,555,555,555
BEGIN DESCRIPTION:
PEACH CREEK9137
END DESCRIPTION:
XS GIS Cut Line= 5
      2522831.67     13850078.69      2521714.98     13849751.66
        2521675.       13849725.        2521652.       13849702.
      2519731.99     13849233.17
#Sta/Elev= 30
  3784.1  400.21  3999.5  394.44  4447.5  392.26  4616.5  385.88  4708.9  385.97
  4742.3  382.74  4760.1  385.97  4905.5  388.35  4916.7  388.49  4973.2  388.13
  4999.3  381.36  5003.6  377.24  5004.6  376.74  5044.5  377.24  5045.8  385.58
  5056.1  387.78  5150.9  387.51  5200.2  386.88  5354.6  392.52  5560.5  390.25
  5632.5   396.6  5668.8   392.1  5768.4  393.06  5840.6  392.47  5862.7  394.75
  6116.3  402.48  6424.4  416.55  6649.6  426.36  6909.2  440.03  7004.7  443.76
#Mann= 12 ,-1 , 0
  3784.1    .045       0  4616.5      .1       0  4905.5     .05       0
  4916.7      .1       0  5003.6     .05       0  5044.5      .1       0
  5150.9     .05       0  5768.4    .035       0  5862.7     .05       0
  6424.4     .07       0  6649.6     .05       0  6909.2     .07       0
Bank Sta=5003.6,5044.5
XS Rating Curve= 0 ,0
Exp/Cntr=0.3,0.1

Type RM Length L Ch R = 1 ,257085  ,567,567,567
BEGIN DESCRIPTION:
PEACH CREEK9136
END DESCRIPTION:
XS GIS Cut Line= 6
      2523065.34     13849350.25      2521965.23     13849347.77
        2521875.       13849275.      2521853.76     13849255.75
      2521489.29     13849339.15      2519752.74     13849128.99
#Sta/Elev= 30
  3783.5  399.86  3853.8  400.76  4253.8  386.59  4733.8   389.1  4783.8  386.46
    4887  388.43  4942.7  386.66  4964.3  376.61  4965.5  376.07  4966.5  375.57
  5006.4  376.07  5013.4   380.3  5020.8  379.28    5025  381.86  5044.8  382.19
  5049.9  378.86  5087.7  387.48  5092.8  385.52  5119.2  388.56  5228.8  391.18
  5244.5   391.7  5346.2  393.16  5545.6  394.12  5743.4  394.93  6156.6  399.65
  6628.8  418.01  6929.6  432.65  6939.5  433.51    7128  443.69  7151.3  444.65
#Mann= 14 ,-1 , 0
  3783.5    .045       0  4964.3    .035       0  4965.5    .035       0
  5006.4    .035       0  5228.8      .1       0  5244.5     .07       0
  5346.2    .035       0  5545.6     .05       0  5743.4    .035       0
  6156.6     .05       0  6628.8     .07       0  6929.6     .05       0
  6939.5     .07       0    7128     .05       0
Bank Sta=4965.5,5006.4
XS Rating Curve= 0 ,0
Exp/Cntr=0.3,0.1

Type RM Length L Ch R = 1 ,256518  ,523,523,523
BEGIN DESCRIPTION:
PEACH CREEK9135
END DESCRIPTION:
XS GIS Cut Line= 5
      2523211.08     13849066.49      2522318.98     13848973.99
        2522175.       13848875.      2522162.58     13848859.48
      2520093.03     13848288.71
#Sta/Elev= 30
  3932.3  399.02  4059.1  397.25  4307.1  387.42  4451.1  384.89    4612  387.81
  4924.7  387.07  4967.5  384.28  4969.8  377.27  4970.8  376.77  5010.9  377.27
  5011.1  380.45  5023.4  382.73  5063.7  384.99    5343  384.02  5359.4  385.67
  5393.7  382.87  5512.4  387.27  5665.4  386.35  5944.5  394.26  6162.3  394.96
  6454.5  406.06  6556.5  404.91  6660.3  413.89  6732.9  417.02  6774.4  414.48
  6817.9  419.98  7016.7  428.17  7051.1  434.43  7158.7  440.68  7170.6  441.45
#Mann= 7 ,-1 , 0
  3932.3     .05       0  4307.1      .1       0  4969.8     .05       0
  5010.9      .1       0    5343     .12       0  6817.9     .07       0
  7158.7    .035       0
Bank Sta=4969.8,5010.9
XS Rating Curve= 0 ,0
Exp/Cntr=0.3,0.1

Type RM Length L Ch R = 1 ,255995  ,567,567,567
BEGIN DESCRIPTION:
PEACH CREEK9134
END DESCRIPTION:
XS GIS Cut Line= 5
      2523176.42     13849024.84      2522600.58     13848809.11
        2522575.       13848775.      2522543.65     13848736.41
       2520538.9     13847650.58
#Sta/Elev= 30
  4338.1  399.04  4433.9  397.12  4637.7  387.74  4788.1  384.19  4973.8  387.04
  4988.4   380.9  4988.7  374.45  4989.7  373.95  5029.8  374.45  5031.6  379.08
    5038   382.3  5059.9  381.22  5112.1  388.44  5142.2   386.7    5264  386.36
  5339.5  385.88    5595  392.98  5878.7  392.93  6069.9   397.4  6129.8   401.8
  6355.7  404.83  6367.6  405.07  6477.9  406.47  6573.6  408.11  6588.3  408.68
  6698.7  410.84    6903  417.57  7030.5  421.51    7243  433.31  7325.3  437.81
#Mann= 15 ,-1 , 0
  4338.1     .05       0  4637.7      .1       0  4988.7     .05       0
  5029.8      .1       0  5142.2     .12       0    5264    .035       0
    5595     .12       0  6355.7    .035       0  6367.6     .07       0
  6477.9    .035       0  6573.6     .12       0  6588.3    .035       0
  6698.7     .12       0    6903     .07       0    7243     .12       0
Bank Sta=4988.7,5029.8
XS Rating Curve= 0 ,0
Exp/Cntr=0.3,0.1

Type RM Length L Ch R = 1 ,255428  ,576,576,576
BEGIN DESCRIPTION:
PEACH CREEK9133
END DESCRIPTION:
XS GIS Cut Line= 3
      2523175.03     13848975.04        2522675.       13848375.
      2521974.99     13847574.99
#Sta/Elev= 30
  4218.7  398.67  4410.8  393.49  4536.1  387.16  4630.7  383.36  4699.1  383.69
  4793.7  385.39  4943.1  386.38  4971.8  381.61  4972.1  373.86  4973.1  373.36
  5013.2  373.86  5013.5  381.18  5021.1  383.66    5042  387.45    5191   385.8
  5205.3  383.79  5212.4  384.67  5268.8  383.58  5290.7   384.4  5297.3  383.22
  5311.6  385.22  5333.6  385.59  5710.5  392.93  5935.1  397.14  5970.2   398.9
  5978.6  398.16  6006.3  399.89  6027.2  402.75  6034.8  401.31  6062.8  402.93
#Mann= 9 ,-1 , 0
  4218.7     .05       0  4536.1      .1       0  4699.1     .05       0
  4793.7      .1       0  4972.1     .05       0  5013.2      .1       0
  5333.6     .12       0  5710.5     .07       0  5978.6     .12       0
Bank Sta=4972.1,5013.2
XS Rating Curve= 0 ,0
Exp/Cntr=0.3,0.1

Type RM Length L Ch R = 1 ,254852  ,550,550,550
BEGIN DESCRIPTION:
PEACH CREEK9132
END DESCRIPTION:
XS GIS Cut Line= 3
        2523225.     13848974.98        2523175.       13848575.
      2521574.98     13847124.98
#Sta/Elev= 30
    4597  398.56  4909.4  391.47  4939.6  391.04  4949.7  389.74  4957.3  387.03
  4962.3  388.17  4979.9  380.39  4985.9   373.9  4986.9   373.4  5028.5   373.9
  5042.3  384.53  5084.9  385.53  5113.3  384.63  5198.5  386.15  5247.8  384.44
  5488.4  386.33  5630.3  384.74  5785.2  386.25  5936.4  388.31  6087.6   390.8
  6182.5  393.35  6279.4  393.78  6470.7  398.73  6557.5  400.03  6671.1  405.49
  6741.4  407.01  6968.7  418.22  7075.7  423.08  7146.1  425.24  7159.4  426.63
#Mann= 12 ,-1 , 0
    4597     .05       0  4909.4      .1       0  4985.9     .05       0
  5028.5      .1       0  5785.2     .12       0  5936.4    .035       0
  6087.6     .07       0  6279.4    .035       0  6470.7     .12       0
  6968.7     .05       0  7075.7     .12       0  7146.1     .05       0
Bank Sta=4985.9,5028.5
XS Rating Curve= 0 ,0
Exp/Cntr=0.3,0.1

Type RM Length L Ch R = 1 ,254302  ,551,551,551
BEGIN DESCRIPTION:
PEACH CREEK9131
END DESCRIPTION:
XS GIS Cut Line= 3
      2524325.01     13849725.01        2523225.       13848175.
      2521624.98     13847024.99
#Sta/Elev= 30
  3099.2  402.62  3504.7  394.69  3782.8  391.17  3806.5  391.61  4137.9  384.56
  4325.5  388.19  4374.3  388.27  4560.7   386.6  4633.3  388.82  4774.7   384.9
  4805.5   388.1    4914  382.21  4950.7  383.91  4956.8  380.67  4971.6  383.25
    5003  379.21  5006.8  373.99  5007.8  373.49  5049.4  373.99  5057.6  383.76
  5330.2  387.06  5370.5  387.48  5444.2  388.95    5546  389.78    5577  389.66
  5951.8  392.78  6023.6  393.59  6247.7  398.28    6774  419.48  6970.3  425.55
#Mann= 20 ,-1 , 0
  3099.2     .05       0  3504.7    .035       0  3782.8     .07       0
  3806.5      .1       0  4137.9     .12       0  4325.5     .05       0
  4374.3    .035       0  4560.7     .12       0  4774.7      .1       0
  5006.8     .05       0  5049.4      .1       0  5330.2     .12       0
  5370.5     .07       0  5444.2     .12       0    5546     .07       0
    5577    .035       0  5951.8     .07       0  6023.6    .035       0
  6247.7     .12       0    6774     .07       0
Bank Sta=5006.8,5049.4
XS Rating Curve= 0 ,0
Exp/Cntr=0.3,0.1

Type RM Length L Ch R = 1 ,253751  ,1076,1076,1076
BEGIN DESCRIPTION:
PEACH CREEK9130
END DESCRIPTION:
XS GIS Cut Line= 3
      2524374.99     13849424.97        2523575.       13847875.
      2521975.04     13846875.02
#Sta/Elev= 30
  3256.3  397.28  3297.5  396.53  3535.9  392.08  3609.2  390.95  3967.7  388.48
  4228.1  383.06  4346.4  386.85  4386.8  386.98  4434.7  387.65  4615.6  387.54
  4786.7  381.09  4838.1  383.53    4946  383.69  4955.5  381.82  4956.6   370.9
  4957.6   370.4  4999.5   370.9  5000.5  381.83  5023.5  383.96  5196.9   380.4
  5220.8  382.61  5275.9  382.65  5327.8  389.54  5480.4   390.1  5576.6  389.74
    5597  389.51  6061.3  391.97  6278.4  397.13  6733.6  414.32  6887.3  419.45
#Mann= 17 ,-1 , 0
  3256.3     .05       0  3297.5    .035       0  3535.9     .05       0
  3609.2     .07       0  3967.7      .1       0  4346.4     .07       0
  4386.8      .1       0  4434.7     .12       0  4838.1      .1       0
  4956.6     .05       0  4999.5      .1       0  5220.8     .12       0
  5480.4    .035       0  5576.6     .12       0    5597    .035       0
  6278.4     .12       0  6733.6     .07       0
Bank Sta=4956.6,4999.5
XS Rating Curve= 0 ,0
Exp/Cntr=0.3,0.1

Type RM Length L Ch R = 1 ,252675  ,532,532,532
BEGIN DESCRIPTION:
PEACH CREEK9129
END DESCRIPTION:
XS GIS Cut Line= 3
      2526474.98     13848124.99        2524075.       13847525.
      2522775.02     13846825.01
#Sta/Elev= 30
  2534.1  401.62  3070.1  393.17  3421.2  384.65  3513.2  381.63  3606.1  382.88
  3657.6  380.64  3714.9  383.48  3757.2  381.85  3794.2   381.8  3830.3  384.74
  3977.2  385.03  4206.5  389.51  4729.6  389.31  4850.8  387.43  4935.8  383.44
  4948.7  381.21  5010.8  379.56  5016.1  376.23  5016.5  370.22  5017.5  369.72
  5059.4  370.22  5059.9  376.11  5087.4  381.79  5244.7  382.63  5325.9   380.1
  5474.3  384.92  5651.3  388.58    6081   389.4  6250.3  392.93  6484.4  399.86
#Mann= 13 ,-1 , 0
  2534.1     .05       0  3421.2     .07       0  3513.2      .1       0
  3714.9     .07       0  3757.2    .045       0  4850.8      .1       0
  5016.5     .05       0  5059.4      .1       0  5244.7     .12       0
  5474.3     .07       0  5651.3     .12       0    6081     .07       0
  6250.3     .12       0
Bank Sta=5016.5,5059.4
XS Rating Curve= 0 ,0
Exp/Cntr=0.3,0.1

Type RM Length L Ch R = 1 ,252143  ,527,527,527
BEGIN DESCRIPTION:
PEACH CREEK9128
END DESCRIPTION:
XS GIS Cut Line= 3
      2526024.99       13847875.        2524025.       13847075.
      2522875.02       13846825.
#Sta/Elev= 30
  2852.1  395.91  3058.1  392.28  3296.7  383.57  3384.1  381.29  3497.1  381.63
  3513.1  380.52  3519.9   376.4  3552.2  381.66    3594  382.14    4413  390.03
  4643.3  388.84    4816  383.02  4876.9  379.67  4967.1  381.29  4973.8  380.06
    4982  370.09    4983  369.59  5024.9  370.09  5025.6  377.49  5030.7  375.19
  5036.9  379.96  5103.5  380.07  5190.4  380.27  5384.8  387.69  5495.5  387.87
  5495.8  387.86    5695  387.61  5865.8  388.75  6053.5  394.36    6183  398.88
#Mann= 15 ,-1 , 0
  2852.1     .05       0  3296.7     .07       0  3384.1     .12       0
  3497.1     .07       0    3594    .045       0    4413     .05       0
  4643.3     .07       0    4816      .1       0    4982     .05       0
  5024.9      .1       0  5103.5     .12       0  5495.5     .07       0
  5495.8     .12       0    5695     .07       0  6053.5     .12       0
Bank Sta=4982,5024.9
XS Rating Curve= 0 ,0
Exp/Cntr=0.3,0.1

Type RM Length L Ch R = 1 ,251616  ,532,532,532
BEGIN DESCRIPTION:
PEACH CREEK9127
END DESCRIPTION:
XS GIS Cut Line= 3
      2526274.96     13847874.98        2524275.       13846675.
        2522825.       13846725.
#Sta/Elev= 30
  2663.5  400.29  3021.1  396.54  3439.3  382.11  3514.8  377.82  3523.1  380.44
  3636.1   379.9  3705.2  379.99    3749  380.44    3862  384.04  3897.9  385.25
  4389.4  382.93  4595.4  386.46  4864.2  385.17  4988.1  380.29  4992.9  377.47
  4994.4  371.34  4995.4  370.84  5037.4  371.34  5045.9  378.48  5065.9  380.95
    5226  379.75  5275.7  381.57  5366.1  376.09  5446.1  382.57  5533.1  383.58
  5979.1  387.39  6219.3  395.36    6237  396.14  6386.7  402.25  6446.7  402.34
#Mann= 16 ,-1 , 0
  2663.5     .05       0  3439.3     .07       0  3523.1     .12       0
  3636.1     .07       0  3705.2     .12       0    3749     .05       0
    3862    .045       0  3897.9     .05       0  4864.2      .1       0
  4994.4     .05       0  5037.4      .1       0  5275.7     .12       0
  5533.1    .035       0  5979.1     .12       0  6219.3     .07       0
    6237     .12       0
Bank Sta=4994.4,5037.4
XS Rating Curve= 0 ,0
Exp/Cntr=0.3,0.1

Type RM Length L Ch R = 1 ,251084  ,540,540,540
BEGIN DESCRIPTION:
PEACH CREEK9126
END DESCRIPTION:
XS GIS Cut Line= 3
      2525925.03     13847575.03        2524375.       13846175.
        2522925.       13845175.
#Sta/Elev= 30
    2912  393.72  3339.6  381.95  3554.9  379.47  3591.7  375.57  3619.5  379.32
    3685  380.14  3917.5   383.2  4090.3  380.24  4139.2   379.7  4858.1  379.72
  4958.5  379.42  4965.2  378.71  4971.8  368.92  4972.8  368.42  5015.4  368.92
    5023  379.14  5029.1  379.39  5208.3  376.06  5476.1  379.49  5625.1  382.17
    5686  383.73  5889.2  385.45  5986.5   386.5  6038.2  387.65  6155.6  390.34
  6167.1     391    6273  393.79  6528.4  402.29  6625.2  404.68  6762.1  407.31
#Mann= 20 ,-1 , 0
    2912     .05       0  3339.6     .07       0  3554.9      .1       0
    3685     .05       0  4090.3    .035       0  4139.2     .05       0
  4858.1      .1       0  4971.8     .05       0  5015.4      .1       0
  5476.1     .12       0  5625.1    .035       0    5686     .12       0
  5889.2     .07       0  5986.5     .05       0  6038.2     .07       0
  6155.6     .12       0  6167.1     .07       0    6273     .12       0
  6528.4    .035       0  6625.2     .12       0
Bank Sta=4971.8,5015.4
XS Rating Curve= 0 ,0
Exp/Cntr=0.3,0.1

Type RM Length L Ch R = 1 ,250544  ,554,554,554
BEGIN DESCRIPTION:
PEACH CREEK9125
END DESCRIPTION:
XS GIS Cut Line= 3
      2526524.98     13847424.98        2524325.       13845825.
      2523175.02     13845275.01
#Sta/Elev= 30
  2279.7  403.72  3082.2  385.03  3481.8  382.58  3686.8  377.84  3766.9  378.78
  3818.7  377.02  3833.4  373.92  3940.9  375.34    3953  375.85  4083.2  377.48
  4234.2  378.61  4304.5  379.22  4377.5  379.01  4419.2     375  4484.1  379.17
  4736.5  378.57  4963.3  378.73  4964.6  369.44  4965.6  368.94  5008.2  369.44
  5008.5     378  5014.1  379.21  5240.3  380.01    5333  381.38  5610.3  385.05
  5702.8  385.56  5942.3   390.9  6102.3  396.71  6190.3   398.8  6274.7  402.01
#Mann= 18 ,-1 , 0
  2279.7     .05       0  3686.8      .1       0  3766.9    .035       0
  3940.9     .05       0    3953     .07       0  4083.2     .05       0
  4234.2     .12       0  4304.5     .05       0  4736.5      .1       0
  4964.6     .05       0  5008.2      .1       0  5240.3     .12       0
    5333     .05       0  5610.3     .07       0  5702.8     .05       0
  5942.3     .07       0  6102.3     .12       0  6190.3     .05       0
Bank Sta=4964.6,5008.2
XS Rating Curve= 0 ,0
Exp/Cntr=0.3,0.1

Type RM Length L Ch R = 1 ,249990  ,1651,1651,1651
BEGIN DESCRIPTION:
PEACH CREEK9124
END DESCRIPTION:
XS GIS Cut Line= 3
      2526324.97     13847174.97        2524775.       13845625.
      2523174.98     13845074.99
#Sta/Elev= 30
  2802.3  396.42  3283.1  386.06  3792.2  383.16  4061.9  376.91  4063.6  376.88
    4243  374.83  4287.2  375.87  4315.5  369.07  4357.9  376.71  4467.1  377.11
  4626.6  378.33  4739.7  375.23  4815.6   377.9  4821.4  378.31  4909.4  378.86
  4951.9  370.21  4980.1  370.91  4982.8   366.8  4983.8   366.3  5026.5   366.8
  5035.9  377.15  5041.1  375.04  5173.9   374.9  5279.8  379.07  5380.2  377.81
  5483.4  379.46  6056.3  385.75  6391.8  396.79  6566.3  401.66  6686.2  405.94
#Mann= 14 ,-1 , 0
  2802.3     .05       0  4061.9    .035       0  4063.6     .05       0
    4243      .1       0  4467.1     .12       0  4815.6     .05       0
  4821.4      .1       0  4982.8     .05       0  5026.5      .1       0
  5173.9     .12       0  5380.2     .07       0  5483.4     .05       0
  6391.8     .07       0  6566.3     .05       0
Bank Sta=4982.8,5026.5
XS Rating Curve= 0 ,0
Exp/Cntr=0.3,0.1

Type RM Length L Ch R = 1 ,248339  ,1095,1095,1095
BEGIN DESCRIPTION:
PEACH CREEK9123
END DESCRIPTION:
XS GIS Cut Line= 3
      2526574.96     13845724.99        2525825.       13845475.
      2523425.03       13845075.
#Sta/Elev= 30
  4210.5  392.62  4214.5  392.56  4723.3  374.23  4937.8  376.35  4958.9  369.54
  4979.9  370.39  4998.9  364.87  4999.9  364.37  5043.7  364.87    5072  379.53
  5102.4  376.56  5257.4  377.35  5315.5  376.83  5758.8  376.98  5763.9  379.83
  5819.7  377.82  5824.7  380.99  5862.7  378.18  5880.5   373.1  5885.6   377.7
  5903.3  382.28  5941.3  379.01  5964.1  384.05  6039.3  382.39  6129.9   380.9
  6388.5  378.74  6761.1  384.26  6969.8  384.87  7337.2  394.84  7434.1  398.83
#Mann= 13 ,-1 , 0
  4210.5    .035       0  4214.5     .05       0  4723.3      .1       0
  4998.9     .05       0  5043.7      .1       0  5257.4     .07       0
  5315.5      .1       0  6039.3     .05       0  6129.9     .07       0
  6388.5     .05       0  6761.1     .07       0  6969.8     .05       0
  7337.2     .07       0
Bank Sta=4998.9,5043.7
XS Rating Curve= 0 ,0
Exp/Cntr=0.3,0.1

Type RM Length L Ch R = 1 ,247244  ,550,550,550
BEGIN DESCRIPTION:
PEACH CREEK9122
END DESCRIPTION:
XS GIS Cut Line= 3
        2526675.       13845375.        2526075.       13844925.
      2523675.02     13844125.01
#Sta/Elev= 30
  4243.6  391.63  4430.1  385.72  4736.3  379.03    4842  374.42  4893.6   374.2
  4930.1  371.86  4936.3  374.12  4950.9  373.89  4965.5  375.53    4968   369.3
    4969   368.8    5013   369.3  5014.7  372.37  5025.2   375.5  5067.4  373.02
  5077.9  375.12    5236  373.99  5299.3  375.71    5378   375.4  5423.8  376.52
  5474.8  378.14    5563  380.63    5744  381.68  6041.2  383.01  6487.7  382.68
  6782.9  382.62  6818.3  383.69  6952.4  383.12  7259.9  385.72  7523.4  391.27
#Mann= 14 ,-1 , 0
  4243.6     .05       0    4842      .1       0    4968     .05       0
    5013      .1       0    5378     .05       0  5423.8      .1       0
  5474.8     .07       0    5563     .05       0    5744     .07       0
  6041.2     .05       0  6487.7     .07       0  6782.9     .05       0
  6818.3     .07       0  6952.4     .05       0
Bank Sta=4968,5013
XS Rating Curve= 0 ,0
Exp/Cntr=0.3,0.1

Type RM Length L Ch R = 1 ,246694  ,1622,1622,1622
BEGIN DESCRIPTION:
PEACH CREEK9121
END DESCRIPTION:
XS GIS Cut Line= 3
      2527274.98     13845574.99        2525875.       13844475.
      2524275.02     13843475.01
#Sta/Elev= 30
  3230.7  413.64    3679  396.08  4049.5  384.65  4113.7  380.23  4163.4  382.58
  4270.9  381.42  4473.7  371.72  4519.5  368.83  4548.4   374.3  4577.3  375.06
  4925.3  374.37  4933.4  371.86  4939.7  374.04  4946.1  363.49  4947.1  362.99
  4991.1  363.49  4997.5  366.37  5003.9  364.66    5008  368.17  5018.8  370.95
  5061.2  373.05  5105.5   381.8  5145.9  381.95  5302.5  380.61  5667.5  381.22
  5762.1  381.25  5876.2  381.27  6499.2  382.25  6711.8  384.96  6897.9  388.51
#Mann= 11 ,-1 , 0
  3230.7     .05       0  4473.7      .1       0  4946.1     .05       0
  4991.1      .1       0  5145.9     .07       0  5302.5     .05       0
  5667.5     .07       0  5762.1     .05       0  5876.2     .07       0
  6499.2     .05       0  6711.8    .035       0
Bank Sta=4946.1,4991.1
XS Rating Curve= 0 ,0
Exp/Cntr=0.3,0.1

Type RM Length L Ch R = 1 ,245072  ,523,523,523
BEGIN DESCRIPTION:
PEACH CREEK9120
END DESCRIPTION:
XS GIS Cut Line= 3
        2527275.       13844425.        2526625.       13844175.
      2524225.03     13843375.01
#Sta/Elev= 30
  4309.6  385.98  4470.3  381.39  4620.3  381.47  4735.3  378.45  4811.1  377.03
  4854.1  375.32  4912.5     373  4996.4  371.63  5003.3  368.37  5004.5  360.24
  5005.5  359.74  5049.6  360.24  5058.7  372.64    5259  372.39  5353.9  374.84
  5374.9  372.48  5448.7  373.81  5469.8  372.35  5480.4  374.16  5677.9  379.01
    6065  379.15  6228.3  380.66  6460.7  380.16  6481.9  378.23  6518.5  380.56
  6870.1  380.69  7209.9  385.77  7251.2  384.68  7356.6  389.62  7535.8  392.88
#Mann= 14 ,-1 , 0
  4309.6     .05       0  4735.3     .07       0  4811.1      .1       0
  4854.1     .07       0  4912.5      .1       0  5004.5     .05       0
  5049.6      .1       0  5677.9     .07       0    6065     .05       0
  6228.3     .07       0  6481.9     .05       0  6518.5     .07       0
  6870.1    .035       0  7209.9     .05       0
Bank Sta=5004.5,5049.6
XS Rating Curve= 0 ,0
Exp/Cntr=0.3,0.1

Type RM Length L Ch R = 1 ,244549  ,522,522,522
BEGIN DESCRIPTION:
PEACH CREEK9119
END DESCRIPTION:
XS GIS Cut Line= 3
      2527824.99       13844225.        2526425.       13843725.
      2524224.97     13843324.99
#Sta/Elev= 30
  3519.5  401.92  3576.4  400.64  3991.8  385.14  4036.2  384.28  4216.6  380.14
  4426.9  380.44  4689.8   374.5  4867.5  371.43  4898.3  366.11  4903.6  368.14
  4921.1  366.26  4934.4  368.62  4959.9  365.84  4962.3  362.98  4963.3  362.48
  5007.4  362.98  5008.6  365.82  5016.3  369.61  5100.3  372.26  5128.1  370.15
  5168.7  373.03  5399.2  377.49  5636.9  378.16  5727.7  378.61  5868.8  375.91
  6287.4  380.03  6603.1  379.74  6805.1  381.57    7110  391.68  7242.2  393.33
#Mann= 11 ,-1 , 0
  3519.5    .035       0  3576.4     .05       0  3991.8     .07       0
  4036.2     .05       0  4689.8      .1       0  4962.3     .05       0
  5007.4      .1       0  5100.3    .035       0  5399.2     .07       0
  5636.9    .035       0  6287.4     .05       0
Bank Sta=4962.3,5007.4
XS Rating Curve= 0 ,0
Exp/Cntr=0.3,0.1

Type RM Length L Ch R = 1 ,244027  ,576,576,576
BEGIN DESCRIPTION:
PEACH CREEK9118
END DESCRIPTION:
XS GIS Cut Line= 3
        2527775.       13844025.        2526525.       13843375.
      2524324.98       13843175.
#Sta/Elev= 30
  3595.7   398.8  3974.6   385.3  4109.9  382.32  4189.4  379.82  4223.3  379.51
  4414.8  377.81  4521.2  378.65  4640.2  375.12  4722.8  374.45  4770.5  366.55
  4780.9  365.86  4825.1  372.28  4841.6  368.26  4869.3  372.26  4891.9  369.83
    4930  371.01  4959.5   367.4  4968.2  360.01  4969.2  359.51  5013.3  360.01
  5014.6   370.4  5358.9  373.94  5587.8  374.25  5617.1  371.37  5697.4  370.62
  5717.5  373.87  5780.3     376  5878.9  378.34  6781.9  379.92  7213.7  393.02
#Mann= 14 ,-1 , 0
  3595.7     .05       0  3974.6     .07       0  4109.9     .05       0
  4189.4     .07       0  4223.3     .05       0  4414.8    .035       0
  4640.2     .12       0  4770.5      .1       0  4968.2     .05       0
  5013.3      .1       0  5358.9     .12       0  5587.8      .1       0
  5780.3     .12       0  5878.9     .05       0
Bank Sta=4968.2,5013.3
XS Rating Curve= 0 ,0
Exp/Cntr=0.3,0.1

Type RM Length L Ch R = 1 ,243451  ,552,552,552
BEGIN DESCRIPTION:
PEACH CREEK9117
END DESCRIPTION:
XS GIS Cut Line= 3
      2527875.01     13843725.01        2526475.       13842925.
      2524275.04       13843125.
#Sta/Elev= 30
  3387.5  393.39  3796.7  384.58  3908.4  380.81  3920.5  380.78  4518.9  372.41
  4578.4  371.82  4690.1  372.32  4801.8  370.84  4815.7  372.82  4846.6  365.89
  4852.4  369.24  4868.2  364.35  4889.8  368.51  4896.3  365.71  4896.7   358.1
  4897.7   357.6  4941.9   358.1  4948.9  364.54  4954.6  360.36  4976.9   359.8
  4986.3  365.59    4992  362.07  5030.1  368.92  5070.3  370.64  5321.3     367
    5419  373.63  5518.2  375.82  6024.2   382.4  6696.9  379.72    7209  393.11
#Mann= 12 ,-1 , 0
  3387.5    .035       0  3796.7     .05       0  3908.4     .07       0
  3920.5     .05       0  4518.9    .035       0  4578.4      .1       0
  4690.1    .035       0  4801.8      .1       0  4896.7     .05       0
  4941.9      .1       0    5419     .12       0  5518.2     .05       0
Bank Sta=4896.7,4941.9
XS Rating Curve= 0 ,0
Exp/Cntr=0.3,0.1

Type RM Length L Ch R = 1 ,242899  ,1587,1587,1587
BEGIN DESCRIPTION:
PEACH CREEK9116
END DESCRIPTION:
XS GIS Cut Line= 3
      2527725.01     13843275.01        2526175.       13842475.
      2525575.01       13842775.
#Sta/Elev= 30
  3263.5  384.04  3374.2  382.05  3483.5  380.39    3496  380.16  3592.8  378.73
  3722.9  377.82  3920.6  374.79  4041.6  370.86  4185.4  369.74  4213.2  368.23
  4242.6  370.91  4368.3  372.63  4517.7  371.67  4650.7  369.12  4748.1   369.6
  4905.3  371.14  4940.3  369.17  4949.6  366.55  4955.2  367.34  4971.7  362.15
  4976.9  357.78  4977.9  357.28  5022.2  357.78  5030.2  367.74  5066.5  367.77
  5108.9  371.82    5237  373.94  5376.7   379.2  5477.5  381.73  5678.6  382.95
#Mann= 14 ,-1 , 0
  3263.5     .05       0  3374.2    .035       0  3483.5     .07       0
    3496    .035       0  3592.8     .07       0  3722.9    .035       0
  3920.6     .05       0  4748.1      .1       0  4976.9     .05       0
  5022.2      .1       0  5108.9     .12       0    5237     .05       0
  5376.7     .12       0  5477.5     .05       0
Bank Sta=4976.9,5022.2
XS Rating Curve= 0 ,0
Exp/Cntr=0.3,0.1

Type RM Length L Ch R = 1 ,241312  ,1153,1153,1153
BEGIN DESCRIPTION:
B19970
END DESCRIPTION:
XS GIS Cut Line= 4
      2528738.71     13843041.98      2527131.24     13841996.15
      2526279.09     13841918.68      2524545.71     13842364.13
#Sta/Elev= 30
  2925.3   382.3    3192  380.37  3213.2  379.51  3757.5  376.96  3972.4  377.39
  4125.9   376.3  4377.2  376.04  4740.3  374.09  4869.4  367.83  4904.3  368.66
  4979.8  367.15  4999.9  362.21  5000.5  354.84  5001.5  354.34  5045.9  354.84
  5050.1   371.3  5060.2  373.24  5080.2   368.1  5100.3  367.04  5166.9  368.68
    5271  370.99    5460  368.35  5491.9  370.86  5672.7  371.98  5827.9  369.43
  6219.2  377.64  6641.6  377.33  6729.4  377.62  6977.4   376.9  7488.4  385.34
#Mann= 16 ,-1 , 0
  2925.3     .05       0    3192     .07       0  3213.2     .05       0
  3757.5     .07       0  3972.4    .035       0  4125.9     .05       0
  4377.2     .07       0  4740.3     .12       0  4904.3      .1       0
  5000.5     .05       0  5045.9      .1       0  5166.9     .12       0
  5827.9     .07       0  6641.6     .05       0  6729.4     .07       0
  6977.4     .05       0
Bank Sta=5000.5,5045.9
XS Rating Curve= 0 ,0
Exp/Cntr=0.3,0.1

Type RM Length L Ch R = 1 ,240159  ,1092,1092,1092
BEGIN DESCRIPTION:
PEACH CREEK9115
END DESCRIPTION:
XS GIS Cut Line= 3
        2528525.       13840425.        2526975.       13841275.
      2524730.48     13842170.16
#Sta/Elev= 30
    3226  386.56  3262.5  384.61  3376.6  378.96  3453.7  375.27  3485.2  373.71
  3602.4  366.56  3669.1   368.4    3705  361.58  3727.8  367.51  3833.1  369.67
  3947.2  372.67  4403.7  374.47    4762  370.93  4816.3  368.42  4936.4  368.66
  4948.1   363.9  4957.3  354.83  4958.3  354.33  5002.8  354.83  5003.2  360.76
  5015.3   366.9  5541.1     367  5619.1  368.59  5760.1  365.06  5849.9  367.62
    6165  373.69  6348.8  375.25  6771.1  376.41  7220.9  377.61  7410.2  381.09
#Mann= 20 ,-1 , 0
    3226     .07       0  3262.5     .12       0  3376.6     .07       0
  3453.7     .12       0  3485.2      .1       0  3833.1     .07       0
  3947.2    .035       0  4403.7     .07       0    4762     .12       0
  4816.3      .1       0  4957.3     .05       0  5002.8      .1       0
  5541.1     .12       0  5619.1      .1       0  5760.1     .12       0
  5849.9     .07       0    6165     .12       0  6348.8     .07       0
  6771.1     .07       0  7220.9     .05       0
Bank Sta=4957.3,5002.8
XS Rating Curve= 0 ,0
Exp/Cntr=0.3,0.1

Type RM Length L Ch R = 1 ,239067  ,1653,1653,1653
BEGIN DESCRIPTION:
PEACH CREEK9114
END DESCRIPTION:
XS GIS Cut Line= 3
      2528524.97     13840075.01        2526125.       13840875.
      2524675.04     13841674.98
#Sta/Elev= 30
  2469.7  394.16  2579.7  387.09  2678.3  382.85  2702.4  381.45  2831.9  370.68
  2870.2  374.13  3028.3  364.01  3038.9  367.03  3102.1   365.5  3154.8  359.08
    3197  365.28  3298.4  365.72  3708.6  371.57  4018.9  372.25  4484.5  365.89
  4946.8  366.78  4999.5  362.49  4999.6   355.5  5000.6     355  5045.1   355.5
  5045.2  364.29  5056.8  366.17  5088.9  361.26  5135.1  364.18    5192  369.19
  5382.4   373.3  5483.5  374.04  6266.7   375.9    6458  379.87  6655.5  383.81
#Mann= 16 ,-1 , 0
  2469.7     .07       0  2579.7     .12       0  2678.3      .1       0
  2702.4     .12       0  2831.9      .1       0  3298.4     .05       0
  3708.6     .07       0  4018.9     .12       0  4484.5      .1       0
  4999.6     .05       0  5045.1      .1       0  5135.1     .12       0
  5382.4     .07       0  5483.5     .12       0  6266.7     .05       0
    6458     .07       0
Bank Sta=4999.6,5045.1
XS Rating Curve= 0 ,0
Exp/Cntr=0.3,0.1

Type RM Length L Ch R = 1 ,237414  ,531,531,531
BEGIN DESCRIPTION:
PEACH CREEK9113
END DESCRIPTION:
XS GIS Cut Line= 3
      2527625.04     13839324.97        2526875.       13839825.
      2523675.02     13842324.99
#Sta/Elev= 30
  4098.7  389.02  4203.8   384.4    4455  371.63  4688.5  362.79  4734.2  356.03
  4776.3  361.63  4797.3  356.51  4806.3  363.33  4956.6  365.02  4971.6  363.97
  4974.3  352.19  4975.3  351.69  5019.9  352.19  5021.8  362.88  5036.3  363.95
  5625.9  365.28  6511.5  373.92  6665.8  374.35  6713.1  374.95  6820.1  374.62
  7352.2  375.03  7491.8  377.39  7576.8  378.48  7605.5  378.79  7745.7  382.36
  7931.3  383.82  8054.2  383.76  8573.3  384.64  8925.6  386.23  9060.9  386.75
#Mann= 20 ,-1 , 0
  4098.7     .05       0  4203.8     .12       0    4455      .1       0
  4688.5      .1       0  4974.3     .05       0  5019.9      .1       0
  5625.9     .05       0  6511.5    .035       0  6665.8     .12       0
  6713.1    .035       0  6820.1     .12       0  7352.2     .05       0
  7491.8     .07       0  7576.8     .05       0  7605.5     .07       0
  7745.7     .07       0  7931.3     .07       0  8054.2     .05       0
  8573.3     .07       0  8925.6     .05       0
Bank Sta=4974.3,5019.9
XS Rating Curve= 0 ,0
Exp/Cntr=0.3,0.1

Type RM Length L Ch R = 1 ,236883  ,551,551,551
BEGIN DESCRIPTION:
PEACH CREEK9112
END DESCRIPTION:
XS GIS Cut Line= 3
      2527425.03     13839224.99        2526625.       13839475.
      2524625.01     13841474.99
#Sta/Elev= 30
  4161.9  383.89  4480.4   368.8  4633.4  363.47  4675.3  355.63  4681.1  360.77
  4696.3  361.63  4727.7  355.55  4778.5  362.34  4978.6  362.65  4989.6  360.77
  4990.8  353.64  4991.8  353.14  5037.7  353.64  5042.5  362.02  5070.8  364.57
  5241.1  363.91  5396.2  368.04  5444.4  368.74  5700.7  370.42  5975.9  368.66
  6797.8  374.34  6933.2  374.02  7068.5  373.49  7259.8  374.15  7411.8  376.85
  7473.3  377.45  7609.9  380.21  7689.8  381.44  7745.2  382.24  7828.5  383.45
#Mann= 17 ,-1 , 0
  4161.9     .12       0  4480.4      .1       0  4990.8     .05       0
  5037.7      .1       0  5241.1     .05       0  5396.2    .035       0
  5444.4     .07       0  5700.7     .05       0  6797.8     .07       0
  6933.2    .035       0  7068.5     .12       0  7259.8     .07       0
  7411.8     .05       0  7473.3     .07       0  7609.9     .05       0
  7689.8     .07       0  7745.2     .05       0
Bank Sta=4990.8,5037.7
XS Rating Curve= 0 ,0
Exp/Cntr=0.3,0.1

Type RM Length L Ch R = 1 ,236332  ,1104,1104,1104
BEGIN DESCRIPTION:
PEACH CREEK9111
END DESCRIPTION:
XS GIS Cut Line= 3
      2527275.03     13839125.01        2526575.       13838975.
      2524575.01     13841374.99
#Sta/Elev= 30
  4284.9  378.22  4640.3  363.92  4811.8  363.65  4898.5  365.47  4959.9  359.86
  4976.1  359.51  4981.2  361.59  4984.5  351.17  4985.5  350.67  5031.4  351.17
  5036.6  357.13  5057.4  360.95  5172.8  364.61  5265.8  363.27  5274.3  363.46
  5566.6  367.58  5666.5  370.07  5920.7  370.65  5963.1  370.54  6321.4  367.88
  6611.4  370.52  6671.6  370.35  7297.3  372.34  7422.4  373.66  7547.6  373.74
    7602  374.89  7637.4  376.11    7923  380.18  8047.7  382.27  8124.9  383.01
#Mann= 20 ,-1 , 0
  4284.9     .12       0  4811.8      .1       0  4984.5     .05       0
  5031.4      .1       0  5172.8     .12       0  5265.8     .07       0
  5274.3     .12       0  5566.6     .07       0  5666.5     .12       0
  5920.7     .07       0  5963.1     .05       0  6611.4     .12       0
  6671.6     .05       0  7297.3     .07       0  7422.4    .035       0
  7547.6     .07       0    7602     .05       0  7637.4     .07       0
    7923     .05       0  8047.7     .05       0
Bank Sta=4984.5,5031.4
XS Rating Curve= 0 ,0
Exp/Cntr=0.3,0.1

Type RM Length L Ch R = 1 ,235228  ,2265,2265,2265
BEGIN DESCRIPTION:
PEACH CREEK9110
END DESCRIPTION:
XS GIS Cut Line= 3
      2527624.97     13838674.99        2526075.       13838175.
      2523875.01     13839374.99
#Sta/Elev= 30
  3363.1  386.46  3688.8  377.23  3961.2  366.31  4048.9   364.7  4151.4  362.24
  4170.8  361.99  4228.1  361.52  4356.3  365.44  4529.4   361.4  4636.3   361.6
  4739.5  362.45  4886.6  360.16  4981.2  362.28  4999.8  359.46  5005.5  360.91
  5014.5  358.89  5021.6  355.25  5027.3  356.89  5041.4  349.93  5042.4  349.43
  5089.1  349.93  5094.2  360.16  5146.9  366.05  5197.9  367.21  5942.4  369.21
  6096.6  370.99  6337.5  370.08  7294.9  373.79  7323.3  373.98  7497.7  376.53
#Mann= 11 ,-1 , 0
  3363.1     .12       0  4048.9      .1       0  4151.4     .07       0
  4170.8     .12       0  4636.3      .1       0  5041.4     .05       0
  5089.1      .1       0  5197.9    .045       0  6337.5     .05       0
  7294.9    .035       0  7323.3     .05       0
Bank Sta=5041.4,5089.1
XS Rating Curve= 0 ,0
Exp/Cntr=0.3,0.1

Type RM Length L Ch R = 1 ,232963  ,530,530,530
BEGIN DESCRIPTION:
PEACH CREEK9109
END DESCRIPTION:
XS GIS Cut Line= 3
      2527474.99       13837625.        2525925.       13836975.
        2523725.       13838775.
#Sta/Elev= 30
  3325.8  385.03  3800.8  366.78  4105.5  362.35  4367.1  362.53  4549.9  357.81
  4555.3  354.96  4614.5  357.28  4708.8  357.95  4732.6  351.82  4756.3  355.61
    4909  357.76  4930.7  353.77  4938.6  347.75  4939.6  347.25  4986.9  347.75
    4992  353.29  5013.7  359.02  5282.3  359.21  5531.1   361.5  5681.3  362.48
  5901.7  360.94  5936.9  364.02  6255.5  367.49  6302.1  367.79  6432.4  368.09
  6562.7  367.78  6646.5  368.03  7364.6  371.45  7485.8  371.63  7849.1  374.27
#Mann= 17 ,-1 , 0
  3325.8     .05       0  4105.5     .07       0  4367.1     .12       0
  4614.5      .1       0  4938.6     .05       0  4986.9      .1       0
  5282.3     .05       0  5531.1     .12       0  5681.3     .05       0
  6255.5    .045       0  6302.1     .05       0  6432.4     .07       0
  6432.4     .05       0  6562.7     .07       0  6646.5     .05       0
  7364.6    .035       0  7485.8     .05       0
Bank Sta=4938.6,4986.9
XS Rating Curve= 0 ,0
Exp/Cntr=0.3,0.1

Type RM Length L Ch R = 1 ,232433  ,1707,1707,1707
BEGIN DESCRIPTION:
PEACH CREEK9108
END DESCRIPTION:
XS GIS Cut Line= 3
      2527924.98     13835375.01        2525525.       13836775.
      2523124.99     13839175.01
#Sta/Elev= 30
  2221.5  393.85  2312.9  391.14  2805.9  378.68  2857.2  377.71  3180.3  371.54
  3958.6  362.43  4144.9  360.85  4176.6  360.71  4315.1  360.25  4750.5  359.93
  4949.1  358.96  4964.8  358.12    4968  349.61    4969  349.11  5016.3  349.61
  5028.3  357.43  5125.4  357.92  5410.1  361.22  5523.2  356.95  5593.9  357.08
  5761.8  360.26  5865.6   361.7  5932.8  363.59  6131.3  367.78    6499  364.85
  6761.2  368.53  6991.9  369.33  7158.1  371.26  7842.5  375.87  8394.1   383.1
#Mann= 18 ,-1 , 0
  2221.5     .07       0  2312.9     .05       0  2805.9    .035       0
  2857.2     .05       0  3958.6    .035       0  4144.9     .05       0
  4176.6    .035       0  4315.1     .05       0  4750.5      .1       0
    4968     .05       0  5016.3      .1       0  5125.4     .05       0
  5761.8     .07       0  5865.6     .05       0  5932.8     .07       0
  6761.2     .05       0  6991.9    .035       0  7158.1     .05       0
Bank Sta=4968,5016.3
XS Rating Curve= 0 ,0
Exp/Cntr=0.3,0.1

Type RM Length L Ch R = 1 ,230726  ,534,534,534
BEGIN DESCRIPTION:
PEACH CREEK9107
END DESCRIPTION:
XS GIS Cut Line= 3
      2526375.02       13835975.        2524575.       13836375.
      2522974.98     13837175.01
#Sta/Elev= 30
  3146.6  373.42  3217.9  371.36    3229  371.01  3434.4  364.28    4063  364.17
  4580.8   363.9  4794.4  359.62    4896  356.57  4971.3  355.89    4988  350.48
  4988.5  344.12  4989.5  343.62  5037.2  344.12    5080  354.16    5151   350.5
  5183.4  357.86  5451.7  363.37  5513.2  361.37  5616.6  366.54  5675.3  361.45
  5692.1  366.38    5720  367.65  5749.1   363.6  5831.8  359.43  5848.6  363.68
  5907.3  366.05  6192.5  367.55  6491.2  373.82  6699.5  378.57  6779.4  381.85
#Mann= 14 ,-1 , 0
  3146.6     .05       0  3217.9     .12       0    3229     .05       0
  3434.4     .12       0    4063     .05       0  4794.4    .035       0
    4896      .1       0  4988.5     .05       0  5037.2      .1       0
    5151     .12       0  5749.1     .07       0  6192.5     .05       0
  6491.2    .035       0  6699.5     .12       0
Bank Sta=4988.5,5037.2
XS Rating Curve= 0 ,0
Exp/Cntr=0.3,0.1

Type RM Length L Ch R = 1 ,230192  ,565,565,565
BEGIN DESCRIPTION:
PEACH CREEK9106
END DESCRIPTION:
XS GIS Cut Line= 3
      2527257.14      13835469.5        2524475.       13835875.
      2522875.02     13835325.01
#Sta/Elev= 30
  2188.8  377.25  2330.7  374.57  2457.7   371.7    2616  369.48  2663.1   369.5
  2845.7  368.05  3012.5  368.31  3363.2  371.88  3777.5  364.87  4141.4  365.68
  4535.5  363.08  4791.5  358.53  4891.5  357.05  4970.4  356.93  4990.2  350.68
  4991.6  343.87  4992.6  343.37  5040.3  343.87  5041.9   353.3  5063.8  355.85
  5254.1  357.49  5291.8  362.76  5328.2  357.18  5433.9  353.72  5661.5  363.46
  5966.9  364.54  6244.5  365.96  6438.4  370.92  6463.2  367.57  6692.2  380.06
#Mann= 13 ,-1 , 0
  2188.8    .035       0  2330.7     .07       0  2457.7     .05       0
    2616     .07       0  2663.1     .05       0  2845.7     .07       0
  3012.5     .05       0  4791.5    .035       0  4891.5      .1       0
  4991.6     .05       0  5040.3      .1       0  5328.2     .07       0
  5966.9     .05       0
Bank Sta=4991.6,5040.3
XS Rating Curve= 0 ,0
Exp/Cntr=0.3,0.1

Type RM Length L Ch R = 1 ,229627  ,519,519,519
BEGIN DESCRIPTION:
PEACH CREEK9105
END DESCRIPTION:
XS GIS Cut Line= 3
      2527131.22     13835169.32        2524375.       13835375.
        2522775.       13835275.
#Sta/Elev= 30
    2241  377.21  2307.6     376  2421.3  374.75  2703.5  370.68  2776.8  370.24
  2922.7  369.33  3187.8  365.48  3300.2  366.43  3711.3  363.45  4433.3  363.66
  4782.4   357.2  4924.7  355.22  4964.8  356.22  4970.5  343.88  4971.5  343.38
  5019.3  343.88  5024.9  354.31    5045  356.57  5295.4  356.19  5353.5  359.04
  5473.2  361.75  5571.7  362.96  5706.2  361.62  5893.2   363.6    6097  365.29
  6187.2  368.28  6247.3  364.66  6437.7  375.85  6530.4  383.38    6608  385.69
#Mann= 13 ,-1 , 0
    2241    .035       0  2307.6     .05       0  2421.3     .07       0
  2703.5     .05       0  2776.8     .07       0  2922.7     .05       0
  4782.4      .1       0  4970.5     .05       0  5019.3      .1       0
  5353.5    .035       0  5473.2     .05       0  5571.7     .07       0
  5893.2     .05       0
Bank Sta=4970.5,5019.3
XS Rating Curve= 0 ,0
Exp/Cntr=0.3,0.1

Type RM Length L Ch R = 1 ,229108  ,544,544,544
BEGIN DESCRIPTION:
PEACH CREEK9104
END DESCRIPTION:
XS GIS Cut Line= 3
      2526325.02       13834575.        2524125.       13834975.
      2522824.98       13835175.
#Sta/Elev= 30
  2763.4  379.49  3566.2  363.65  3667.7  362.16  3861.1  358.23  4073.3  362.62
  4206.4  361.84  4355.5  359.41  4362.2  359.47  4506.4  356.88    4584  355.27
  4655.9  356.56  4704.7  354.83  4972.8  355.71  4979.2  353.19  4985.2  343.05
  4986.2  342.55    5034  343.05    5040  354.28  5049.3  354.11  5080.4  356.68
  5879.7  365.27  5930.3  366.27  5949.3  369.93  5960.7     370    5991  361.75
  6001.1     361  6031.5  367.72  6122.5  371.86  6203.5  379.72  6314.8  385.71
#Mann= 11 ,-1 , 0
  2763.4     .05       0  3566.2     .07       0  3667.7     .05       0
  4206.4     .07       0  4355.5     .05       0  4362.2     .07       0
  4506.4     .12       0  4655.9      .1       0  4985.2     .05       0
    5034      .1       0  5049.3     .05       0
Bank Sta=4985.2,5034
XS Rating Curve= 0 ,0
Exp/Cntr=0.3,0.1
