--- SAUL CREEK.prj (project) ---

Proj Title=SAUL CREEK Base Level Engineering
Current Plan=p01
Default Exp/Contr=0.3,0.1
English Units
Geom File=g01
Flow File=f01
Plan File=p01
Y Axis Title=Elevation
X Axis Title(PF)=Main Channel Distance
X Axis Title(XS)=Station
BEGIN DESCRIPTION:
SAUL CREEK
END DESCRIPTION:
DSS Export Rating Curves= 0
DSS Export Rating Curve Sorted= 0
DSS Export Volume Flow Curves= 0
DXF OffsetX= 0
DXF OffsetY= 0
DXF ScaleX= 1
DXF ScaleY= 10

--- SAUL CREEK.p01 (plan) ---

Plan Title=Multiple Run
Short Identifier=Multiple
Geom File=g01
Flow File=f01
Subcritical Flow
K Sum by GR= 0
Std Step Tol= 0.01
Critical Tol= 0.01
Num of Std Step Trials= 20
Max Error Tol= 0.3
Flow Tol Ratio= 0.001
Split Flow NTrial= 30
Split Flow Tol= 0.02
Split Flow Ratio= 0.02
Log Output Level= 0
Friction Slope Method= 1
Unsteady Friction Slope Method= 2
Unsteady Bridges Friction Slope Method= 1
Parabolic Critical Depth
Global Vel Dist=  1 , 1 , 1
Global Log Level= 0
CheckData=True
Encroach Param= -1, 0, 0, 0
BEGIN DESCRIPTION:
Multiple Run
END DESCRIPTION:

--- SAUL CREEK.f01 (steady flow) ---

Flow Title=Multiple
Number of Profiles=7
Profile Names=10-year,25-year,50-year,1pct_min,100-year,1pct_plu,500-year
River Rch & RM= SAUL CREEK,Reach-1,29824
     368     569     742     469     936    1868    1476
River Rch & RM= SAUL CREEK,Reach-1,27062
     852    1381    1859    1209    2413    4815    4031
River Rch & RM= SAUL CREEK,Reach-1,17815
    1150    1898    2586    1702    3395    6774    5803
River Rch & RM= SAUL CREEK,Reach-1,13642
    1858    3141    4351    2906    5798   11569   10215
River Rch & RM= SAUL CREEK,Reach-1,5964
    2222    3787    5273    3539    7060   14087   12558
Boundary for River Rch & Prof#=SAUL CREEK,Reach-1,1
Up Type=0
Dn Type=3
Dn Slope=0.005
Boundary for River Rch & Prof#=SAUL CREEK,Reach-1,2
Up Type=0
Dn Type=3
Dn Slope=0.005
Boundary for River Rch & Prof#=SAUL CREEK,Reach-1,3
Up Type=0
Dn Type=3
Dn Slope=0.005
Boundary for River Rch & Prof#=SAUL CREEK,Reach-1,4
Up Type=0
Dn Type=3
Dn Slope=0.005
Boundary for River Rch & Prof#=SAUL CREEK,Reach-1,5
Up Type=0
Dn Type=3
Dn Slope=0.005
Boundary for River Rch & Prof#=SAUL CREEK,Reach-1,6
Up Type=0
Dn Type=3
Dn Slope=0.005
Boundary for River Rch & Prof#=SAUL CREEK,Reach-1,7
Up Type=0
Dn Type=3
Dn Slope=0.005

--- SAUL CREEK.g01 (geometry) ---

Geom Title=Existing Conditions

River Reach=SAUL CREEK,Reach-1
Reach XY= 30
      2319425.00     13758425.00      2318975.61     13756964.38
      2319025.95     13756135.41      2319823.42     13753968.95
      2319678.34     13753676.72      2320141.40     13753108.25
      2321050.00     13752924.60      2321964.49     13753123.80
      2322823.75     13752971.55      2323135.29     13752626.00
      2323769.31     13752773.13      2323874.75     13752531.98
      2325444.89     13752925.11      2328425.00     13752825.00
      2328674.64     13752509.82      2328578.82     13751676.58
      2329073.51     13751219.15      2328878.75     13750776.55
      2329335.17     13749815.32      2329855.24     13749695.63
      2330030.40     13748972.57      2330519.59     13748627.71
      2330433.00     13748068.67      2330931.05     13747726.67
      2331769.66     13747727.74      2331628.09     13747076.65
      2332474.76     13746009.79      2332176.96     13744730.66
      2332848.86     13744351.93      2332825.00     13744075.00

Type RM Length L Ch R = 1,29824,375,375,375
BEGIN DESCRIPTION:
SAUL CREEK 65.0
END DESCRIPTION:
XS GIS Cut Line= 3
      2319847.22     13758343.33      2319423.73     13758359.42
      2318785.78     13758455.91
#Sta/Elev= 30
  4577.5  519.87  4581.1  519.87  4589.7  518.94  4599.7  518.79  4669.8  518.00
  4699.8  517.98  4719.8  517.51  4769.9  517.30  4809.9  516.42  4920.0  514.87
  4996.2  514.50  4996.4  514.00  4999.9  514.00  5000.2  514.50  5020.2  515.00
  5111.3  515.64  5131.5  516.31  5137.7  516.85  5206.6  517.10  5232.6  517.80
  5303.4  518.83  5354.0  520.36  5364.1  520.15  5408.0  520.50  5455.1  521.99
  5515.8  522.44  5566.4  524.30  5596.7  523.87  5627.1  524.48  5646.5  524.28
#Mann=3,-1,0
  4577.5    0.05       0  4996.2    0.05       0  5000.2    0.05       0
Bank Sta=4996.2,5000.2
Exp/Cntr=0.3,0.1

Type RM Length L Ch R = 1,29449,475,475,475
BEGIN DESCRIPTION:
E20755
END DESCRIPTION:
XS GIS Cut Line= 3
      2319847.23     13757951.97      2319107.43     13758048.47
      2318651.74     13758187.86
#Sta/Elev= 30
  4468.8  517.22  4481.1  516.46  4491.2  516.77  4528.7  516.12  4652.6  515.79
  4765.7  514.56  4894.6  514.22  4945.0  514.57  4990.6  513.36  4990.8  512.86
  4994.3  512.86  4994.6  513.36  5039.2  514.12  5086.2  515.02  5145.5  515.13
  5187.1  516.58  5238.3  516.93  5301.1  518.28  5324.9  517.74  5357.7  518.95
  5390.5  519.26  5423.3  520.85  5456.1  521.14  5468.4  520.73  5520.7  522.42
  5541.6  522.11  5614.8  522.71  5656.6  523.78  5668.4  524.87  5691.4  524.36
#Mann=5,-1,0
  4468.8    0.05       0  4945.0    0.07       0  4990.6    0.07       0
  4994.6    0.07       0  5039.2    0.05       0
Bank Sta=4990.6,4994.6
Exp/Cntr=0.3,0.1

Type RM Length L Ch R = 1,28974,258,258,258
BEGIN DESCRIPTION:
SAUL CREEK 64.0
END DESCRIPTION:
XS GIS Cut Line= 3
      2319875.01     13757325.00      2319080.62     13757742.88
      2318549.92     13757919.78
#Sta/Elev= 30
  4370.6  524.02  4443.2  522.63  4467.0  522.25  4472.6  521.20  4483.3  521.55
  4489.0  520.39  4498.7  520.69  4505.4  520.89  4511.0  519.71  4549.5  519.48
  4555.1  518.54  4703.7  515.70  4852.4  513.69  4890.4  514.08  4940.5  512.79
  4962.6  511.32  4984.6  512.66  5021.0  510.75  5021.3  510.25  5025.0  510.75
  5067.1  512.05  5072.7  513.23  5089.1  513.35  5094.8  514.38  5149.6  512.92
  5229.3  513.27  5669.8  520.23  5695.8  521.57  5727.4  521.06  5827.6  522.19
#Mann=5,-1,0
  4370.6   0.035       0  4443.2   0.063       0  4498.7   0.035       0
  5021.0   0.035       0  5025.0   0.035       0
Bank Sta=5021,5025
Exp/Cntr=0.3,0.1

Type RM Length L Ch R = 1,28716,337,337,337
BEGIN DESCRIPTION:
SAUL CREEK 63.0
END DESCRIPTION:
XS GIS Cut Line= 3
      2319475.03     13757324.99      2318957.31     13757460.89
      2318533.80     13757686.05
#Sta/Elev= 30
  4741.0  517.09  4989.2  511.02  5007.8  506.89  5008.1  506.39  5011.6  506.39
  5011.8  506.89  5020.2  507.47  5030.5  510.88  5036.1  511.83  5071.3  510.97
  5076.4  511.44  5111.6  510.20  5192.4  511.81  5247.6  511.68  5334.1  513.52
  5356.0  513.29  5437.4  514.47  5570.1  517.81  5575.8  516.59  5607.3  518.17
  5630.0  517.04  5636.1  517.34  5641.7  518.50  5652.4  517.82  5658.0  519.60
  5674.4  519.08  5680.0  520.11  5696.3  519.93  5702.0  520.51  5755.9  521.29
#Mann=3,-1,0
  4741.0   0.035       0  5007.8   0.035       0  5011.8   0.035       0
Bank Sta=5007.8,5011.8
Exp/Cntr=0.3,0.1

Type RM Length L Ch R = 1,28379,433,433,433
BEGIN DESCRIPTION:
SAUL CREEK 62.0
END DESCRIPTION:
XS GIS Cut Line= 3
      2319474.96     13757175.00      2319025.00     13757125.00
      2318575.01     13757374.99
#Sta/Elev= 30
  4555.0  517.71  4675.7  514.86  4695.8  513.89  4736.1  513.68  4766.3  512.55
  4816.6  511.38  4947.4  508.88  4985.6  506.91  4985.9  506.41  4989.4  506.41
  4989.6  506.91  5005.2  508.06  5021.5  508.45  5030.6  508.09  5053.5  508.15
  5064.9  508.94  5087.8  509.12  5097.0  509.95  5156.4  510.94  5178.2  511.75
  5183.9  511.44  5227.4  511.86  5259.4  513.27  5281.1  513.63  5293.7  513.02
  5308.6  513.19  5330.3  514.24  5352.1  515.94  5373.8  516.62  5522.5  517.34
#Mann=3,-1,0
  4555.0    0.05       0  4985.6    0.05       0  4989.6    0.05       0
Bank Sta=4985.6,4989.6
Exp/Cntr=0.3,0.1

Type RM Length L Ch R = 1,27946,434,434,434
BEGIN DESCRIPTION:
SAUL CREEK 61.0
END DESCRIPTION:
XS GIS Cut Line= 3
      2319375.03     13756825.00      2319075.00     13756775.00
      2318625.00     13757075.00
#Sta/Elev= 30
  4695.9  513.63  4706.1  513.23  4736.5  513.39  4756.8  512.40  4797.3  511.08
  4858.1  509.84  4878.4  509.48  4888.5  509.66  4911.4  509.00  4939.2  509.31
  4949.4  508.96  4959.5  507.04  4967.1  503.41  4970.2  502.86  4970.4  502.36
  4973.9  502.36  4974.2  502.86  4979.8  505.09  4997.5  506.78  5036.1  506.81
  5043.6  507.26  5085.7  507.83  5094.7  508.26  5130.8  507.80  5151.8  508.13
  5208.9  509.83  5229.9  509.69  5238.9  510.15  5360.6  511.11  5540.9  514.11
#Mann=3,-1,0
  4695.9    0.05       0  4970.2    0.05       0  4974.2    0.05       0
Bank Sta=4970.2,4974.2
Exp/Cntr=0.3,0.1

Type RM Length L Ch R = 1,27512,450,450,450
BEGIN DESCRIPTION:
SAUL CREEK 60.0
END DESCRIPTION:
XS GIS Cut Line= 3
      2319375.02     13756575.01      2319075.00     13756375.00
      2318475.00     13756875.00
#Sta/Elev= 30
  4639.9  512.73  4653.4  512.94  4683.5  511.57  4734.6  510.17  4848.7  508.81
  4940.3  506.87  4964.4  505.66  4971.9  502.63  4975.9  502.07  4976.2  501.57
  4979.7  501.57  4979.9  502.07  4987.0  504.95  4997.5  505.85  5028.5  505.91
  5036.3  506.66  5042.8  506.68  5092.2  505.94  5199.0  508.60  5229.4  508.44
  5369.5  509.49  5391.0  509.26  5554.4  511.69  5632.5  511.90  5653.3  512.37
  5681.9  511.94  5696.2  512.56  5745.7  512.82  5760.0  513.49  5781.5  513.29
#Mann=5,-1,0
  4639.9    0.05       0  4940.3    0.07       0  4975.9    0.07       0
  4979.9    0.07       0  5229.4    0.05       0
Bank Sta=4975.9,4979.9
Exp/Cntr=0.3,0.1

Type RM Length L Ch R = 1,27062,465,465,465
BEGIN DESCRIPTION:
SAUL CREEK 59.0
END DESCRIPTION:
XS GIS Cut Line= 3
      2319574.96     13756174.98      2319175.00     13756025.00
      2318525.02     13755575.01
#Sta/Elev= 30
  4567.9  514.79  4685.3  511.95  4698.7  510.92  4723.6  510.25  4738.7  510.64
  4802.1  509.40  4839.3  508.55  4924.7  504.67  4973.7  504.13  4985.3  499.53
  4990.0  499.30  4990.4  498.80  4994.4  498.80  4994.7  499.30  4998.1  499.30
  5008.6  502.55  5023.4  503.99  5089.0  505.02  5153.2  504.97  5241.3  506.02
  5432.9  508.38  5491.7  510.20  5518.7  510.18  5605.2  512.47  5641.0  514.28
  5664.0  514.01  5691.7  515.30  5741.7  516.38  5757.2  517.41  5785.6  517.22
#Mann=5,-1,0
  4567.9    0.05       0  4802.1    0.12       0  4990.0    0.07       0
  4994.7    0.12       0  5241.3    0.07       0
Bank Sta=4990,4994.7
Exp/Cntr=0.3,0.1

Type RM Length L Ch R = 1,26597,451,451,451
BEGIN DESCRIPTION:
SAUL CREEK 58.0
END DESCRIPTION:
XS GIS Cut Line= 3
      2319674.98     13755924.98      2319275.00     13755625.00
      2318725.02     13755375.01
#Sta/Elev= 30
  4495.8  514.72  4545.8  513.54  4582.2  511.81  4588.5  512.17  4649.5  510.74
  4683.0  509.74  4924.7  505.20  4989.6  502.62  4998.5  502.03  5004.6  499.67
  5015.4  498.33  5015.7  497.83  5019.8  497.83  5020.1  498.33  5027.6  502.01
  5039.7  503.35  5072.7  503.22  5107.8  502.02  5154.0  502.81  5161.1  503.83
  5182.5  503.56  5215.5  504.72  5233.6  504.71  5287.0  505.58  5326.4  506.43
  5441.7  510.91  5493.4  511.22  5556.0  513.16  5578.0  514.49  5599.9  514.31
#Mann=10,-1,0
  4495.8    0.05       0  4649.5    0.07       0  4683.0    0.05       0
  4924.7    0.07       0  4989.6    0.12       0  5015.4    0.07       0
  5020.1    0.12       0  5161.1    0.07       0  5233.6    0.12       0
  5287.0    0.07       0
Bank Sta=5015.4,5020.1
Exp/Cntr=0.3,0.1

Type RM Length L Ch R = 1,26146,486,486,486
BEGIN DESCRIPTION:
SAUL CREEK 57.0
END DESCRIPTION:
XS GIS Cut Line= 3
      2320024.98     13755824.99      2319225.00     13755225.00
      2318824.99     13755175.00
#Sta/Elev= 30
  4004.4  521.44  4032.5  521.01  4040.8  520.24  4090.8  519.65  4138.5  518.04
  4211.7  515.40  4297.1  513.92  4340.8  512.29  4367.9  512.02  4476.3  508.98
  4661.7  505.30  4740.8  504.53  4793.4  503.40  4867.9  503.44  4917.9  502.22
  4932.5  502.46  4990.8  501.84  4997.1  499.68  4998.9  497.30  4999.2  496.80
  5003.3  496.80  5003.7  497.30  5014.5  497.81  5024.5  501.65  5034.6  501.15
  5109.8  505.35  5276.5  509.13  5326.9  511.17  5347.0  511.38  5407.5  513.39
#Mann=6,-1,0
  4004.4    0.05       0  4138.5    0.07       0  4793.4    0.12       0
  4998.9    0.07       0  5003.7    0.12       0  5109.8    0.07       0
Bank Sta=4998.9,5003.7
Exp/Cntr=0.3,0.1

Type RM Length L Ch R = 1,25660,461,461,461
BEGIN DESCRIPTION:
SAUL CREEK 56.0
END DESCRIPTION:
XS GIS Cut Line= 3
      2320074.97     13754875.00      2319425.00     13754825.00
      2319025.00     13754475.00
#Sta/Elev= 30
  4363.3  516.53  4373.3  517.05  4383.3  516.62  4403.4  513.61  4423.4  511.56
  4463.6  509.69  4674.2  504.47  4850.2  501.70  4948.8  500.59  4985.1  500.04
  5022.3  501.01  5029.0  495.91  5036.5  496.68  5040.7  495.11  5041.1  494.61
  5045.7  495.11  5050.3  497.64  5057.4  500.84  5100.1  500.96  5184.3  503.00
  5185.1  503.02  5312.7  505.31  5409.3  508.81  5440.4  508.36  5468.4  508.97
  5476.0  510.06  5482.6  510.08  5496.9  508.98  5518.7  510.38  5546.7  511.13
#Mann=9,-1,0
  4363.3    0.07       0  4850.2    0.12       0  4948.8    0.12       0
  5040.7    0.07       0  5045.7    0.12       0  5050.3    0.05       0
  5184.3    0.12       0  5185.1   0.035       0  5409.3    0.07       0
Bank Sta=5040.7,5045.7
Exp/Cntr=0.3,0.1

Type RM Length L Ch R = 1,25199,479,479,479
BEGIN DESCRIPTION:
SAUL CREEK 55.0
END DESCRIPTION:
XS GIS Cut Line= 3
      2320075.02     13754725.01      2319575.00     13754425.00
      2318975.02     13754425.00
#Sta/Elev= 30
  4420.8  515.32  4431.9  516.25  4444.2  515.24  4455.8  512.43  4465.5  511.29
  4545.2  507.54  4579.4  506.89  4698.8  502.58  4720.1  502.69  4778.5  497.79
  4792.7  497.77  4825.1  497.78  4852.3  500.13  4873.7  504.31  4887.3  503.41
  4900.9  500.79  4910.6  500.10  4964.3  498.50  4980.6  498.07  4987.8  496.24
  4988.2  495.74  4992.8  496.24  5023.9  499.29  5053.9  498.90  5301.0  504.58
  5477.0  509.44  5493.9  508.68  5523.9  510.46  5595.8  512.13  5603.9  512.27
#Mann=11,-1,0
  4420.8    0.07       0  4431.9    0.05       0  4579.4    0.07       0
  4792.7    0.05       0  4825.1    0.07       0  4964.3    0.05       0
  4987.8    0.05       0  4992.8    0.05       0  5301.0   0.035       0
  5477.0    0.07       0  5595.8   0.035       0
Bank Sta=4987.8,4992.8
Exp/Cntr=0.3,0.1

Type RM Length L Ch R = 1,24720,420,420,420
BEGIN DESCRIPTION:
SAUL CREEK 54.0
END DESCRIPTION:
XS GIS Cut Line= 3
      2320174.96     13754224.98      2319775.00     13754025.00
      2318975.03     13753975.00
#Sta/Elev= 30
  4553.1  510.93  4606.2  508.60  4634.1  509.66  4650.9  507.94  4723.6  506.09
  4740.3  504.80  4785.0  503.03  4880.1  500.89  4910.8  498.92  4933.2  498.58
  4963.9  496.98  4969.5  496.49  4975.4  493.79  4975.8  493.29  4980.1  493.29
  4980.5  493.79  4986.3  495.25  4991.9  497.51  4997.5  498.09  5180.6  497.77
  5351.0  501.48  5431.1  502.05  5525.5  504.72  5621.5  507.38  5631.5  508.37
  5651.5  508.03  5661.6  509.19  5681.6  508.73  5741.7  510.49  5801.8  513.18
#Mann=4,-1,0
  4553.1    0.05       0  4975.4    0.05       0  4980.5    0.05       0
  5525.5   0.035       0
Bank Sta=4975.4,4980.5
Exp/Cntr=0.3,0.1

Type RM Length L Ch R = 1,24300,471,471,471
BEGIN DESCRIPTION:
SAUL CREEK 53.0
END DESCRIPTION:
XS GIS Cut Line= 3
      2320375.03     13754275.02      2319675.00     13753675.00
      2319174.98     13753725.00
#Sta/Elev= 30
  4082.0  516.49  4117.5  515.58  4152.8  514.84  4181.4  513.29  4294.4  511.15
  4330.6  508.71  4358.6  509.71  4380.0  508.06  4472.2  505.78  4486.5  504.81
  4500.8  505.62  4578.7  502.22  4755.4  498.19  4777.3  496.90  4968.3  496.86
  4996.9  495.58  4998.0  493.90  4998.5  493.40  5003.3  493.90  5014.0  495.19
  5064.3  497.57  5225.1  501.92  5325.6  502.80  5345.7  503.79  5353.2  504.82
  5358.2  503.98  5375.8  505.50  5445.1  507.85  5466.3  509.45  5506.5  510.12
#Mann=5,-1,0
  4082.0   0.035       0  4117.5    0.05       0  4998.0    0.05       0
  5003.3    0.05       0  5445.1   0.035       0
Bank Sta=4998,5003.3
Exp/Cntr=0.3,0.1

Type RM Length L Ch R = 1,23829,463,463,463
BEGIN DESCRIPTION:
SAUL CREEK 52.0
END DESCRIPTION:
XS GIS Cut Line= 3
      2320425.02     13754075.04      2320025.00     13753425.00
      2319324.99     13752874.99
#Sta/Elev= 30
  4236.8  514.38  4295.6  513.09  4354.0  510.84  4418.5  508.69  4433.9  509.36
  4455.2  507.65  4476.5  507.19  4506.9  505.44  4528.6  506.07  4549.8  504.52
  4681.2  501.19  4855.1  497.37  4906.1  497.10  4964.8  494.54  5003.2  494.72
  5011.0  494.07  5011.4  493.57  5015.9  493.57  5016.3  494.07  5028.1  495.37
  5114.5  495.18  5241.7  498.96  5307.8  499.90  5419.7  502.29  5442.0  503.41
  5527.0  504.48  5544.1  505.49  5576.7  505.54  5705.0  507.94  5890.3  512.66
#Mann=6,-1,0
  4236.8   0.035       0  4354.0    0.05       0  5011.0    0.05       0
  5016.3    0.05       0  5307.8    0.07       0  5544.1   0.035       0
Bank Sta=5011,5016.3
Exp/Cntr=0.3,0.1

Type RM Length L Ch R = 1,23366,443,443,443
BEGIN DESCRIPTION:
SAUL CREEK 51.0
END DESCRIPTION:
XS GIS Cut Line= 3
      2320574.98     13753624.97      2320175.00     13753075.00
      2319675.03     13752575.03
#Sta/Elev= 30
  4319.7  512.48  4322.8  512.48  4327.0  510.12  4333.2  511.32  4341.7  507.64
  4477.7  504.16  4720.4  494.37  4818.1  493.54  4818.6  493.04  4823.5  493.54
  4863.7  495.14  4891.9  499.62  4906.6  500.22  4936.0  499.72  4942.2  497.57
  4956.8  497.86  4963.0  496.75  4971.5  497.88  4977.7  495.96  4984.0  497.11
  4992.4  496.19  4996.6  497.77  5003.3  497.77  5042.2  494.23  5056.3  494.21
  5127.0  495.84  5197.7  499.56  5369.4  501.74  5551.3  505.95  5706.8  511.50
#Mann=5,-1,0
  4319.7    0.05       0  4818.1    0.07       0  4823.5    0.05       0
  4984.0    0.07       0  5369.4   0.035       0
Bank Sta=4818.1,4823.5
Exp/Cntr=0.3,0.1

Type RM Length L Ch R = 1,22923,469,469,469
BEGIN DESCRIPTION:
SAUL CREEK 50.0
END DESCRIPTION:
XS GIS Cut Line= 3
      2320625.00     13753625.03      2320525.00     13752925.00
      2319975.00     13752275.00
#Sta/Elev= 30
  4296.9  508.33  4327.2  508.06  4539.4  502.26  4600.0  499.79  4630.3  499.24
  4711.1  495.27  4791.9  492.95  4832.3  492.24  4953.5  492.24  4983.8  491.86
  4991.2  490.85  4991.6  490.35  4996.2  490.35  4996.6  490.85  5001.5  491.67
  5011.2  492.10  5039.8  491.67  5113.4  492.51  5132.1  492.76  5152.9  493.93
  5186.2  494.86  5195.8  495.38  5245.2  495.16  5252.9  495.77  5292.4  496.70
  5436.3  499.09  5489.4  500.46  5720.9  505.90  5791.2  509.56  5855.5  511.35
#Mann=7,-1,0
  4296.9    0.05       0  4991.2    0.05       0  4996.6    0.05       0
  5113.4    0.07       0  5186.2    0.05       0  5292.4    0.07       0
  5489.4   0.035       0
Bank Sta=4991.2,4996.6
Exp/Cntr=0.3,0.1

Type RM Length L Ch R = 1,22454,480,480,480
BEGIN DESCRIPTION:
SAUL CREEK 49.0
END DESCRIPTION:
XS GIS Cut Line= 3
      2320775.00     13753474.99      2320975.00     13752975.00
      2321174.99     13752425.04
#Sta/Elev= 30
  4455.5  504.04  4524.2  502.38  4572.6  500.13  4638.6  498.96  4763.8  494.50
  4846.8  492.81  4872.7  492.34  4907.8  491.27  4961.7  491.46  4979.2  489.84
  4984.6  490.32  4991.3  489.02  5001.2  488.65  5001.7  488.15  5006.7  488.65
  5009.3  489.85  5081.4  489.87  5105.1  489.84  5156.9  490.60  5182.2  491.99
  5218.1  491.95  5260.0  493.69  5304.6  494.18  5416.3  498.45  5440.9  498.45
  5462.2  500.08  5511.0  501.53  5547.3  502.47  5563.9  503.62  5579.2  503.60
#Mann=8,-1,0
  4455.5    0.05       0  4846.8    0.07       0  4872.7    0.12       0
  5001.2    0.07       0  5006.7    0.12       0  5081.4    0.05       0
  5105.1    0.07       0  5511.0    0.05       0
Bank Sta=5001.2,5006.7
Exp/Cntr=0.3,0.1

Type RM Length L Ch R = 1,21974,445,445,445
BEGIN DESCRIPTION:
SAUL CREEK 48.0
END DESCRIPTION:
XS GIS Cut Line= 3
      2321025.00     13753725.00      2321425.00     13752975.00
      2321475.00     13752524.97
#Sta/Elev= 30
  4149.6  507.68  4198.7  506.60  4223.6  506.48  4289.5  502.93  4423.0  499.12
  4444.3  498.72  4466.9  500.85  4489.6  501.41  4497.7  499.55  4503.4  501.09
  4512.3  499.18  4534.9  498.74  4541.7  497.92  4547.3  498.42  4563.6  496.45
  4601.9  494.82  4735.0  492.36  4857.7  490.36  4887.3  488.60  4947.5  487.89
  4994.0  486.33  4994.4  485.83  4999.5  486.33  5060.0  487.12  5097.1  488.42
  5144.3  491.07  5160.6  492.27  5271.3  496.20  5351.8  500.37  5452.4  503.07
#Mann=9,-1,0
  4149.6    0.07       0  4198.7    0.12       0  4423.0    0.07       0
  4735.0    0.12       0  4857.7    0.05       0  4994.0    0.05       0
  4999.5    0.05       0  5097.1    0.07       0  5144.3    0.05       0
Bank Sta=4994,4999.5
Exp/Cntr=0.3,0.1

Type RM Length L Ch R = 1,21529,459,459,459
BEGIN DESCRIPTION:
SAUL CREEK 47.0
END DESCRIPTION:
XS GIS Cut Line= 3
      2321524.97     13753475.04      2321825.00     13753125.00
      2321574.99     13752574.98
#Sta/Elev= 30
  4532.4  501.77  4553.8  499.72  4568.1  496.92  4582.4  495.22  4742.3  491.90
  4873.2  488.16  4892.7  488.40  4951.2  486.44  4963.4  486.99  4979.7  486.32
  4986.3  485.45  4990.1  483.51  5004.9  482.90  5005.4  482.40  5010.1  482.40
  5010.6  482.90  5036.2  484.11  5082.4  485.25  5158.2  485.72  5180.2  486.25
  5197.7  487.89  5203.2  486.98  5208.4  487.40  5220.8  488.40  5226.3  487.96
  5243.9  489.39  5249.4  488.96  5266.9  490.36  5341.6  493.18  5597.6  501.46
#Mann=8,-1,0
  4532.4    0.07       0  4742.3    0.12       0  4892.7    0.07       0
  4963.4    0.12       0  5004.9    0.07       0  5010.6    0.12       0
  5036.2    0.07       0  5208.4    0.05       0
Bank Sta=5004.9,5010.6
Exp/Cntr=0.3,0.1

Type RM Length L Ch R = 1,21070,466,466,466
BEGIN DESCRIPTION:
SAUL CREEK 46.0
END DESCRIPTION:
XS GIS Cut Line= 3
      2322474.99     13753474.97      2322225.00     13752975.00
      2321874.97     13752624.97
#Sta/Elev= 30
  4440.8  496.42  4461.9  496.59  4471.5  496.68  4485.5  495.49  4516.2  494.56
  4583.3  493.30  4588.9  493.85  4784.6  487.90  4828.8  487.29  4835.3  487.46
  4857.2  487.23  4918.7  484.95  4946.7  485.13  4963.4  484.57  4985.8  482.65
  4994.1  480.26  4994.5  479.76  4999.4  479.76  4999.9  480.26  5013.9  480.93
  5028.1  482.65  5042.2  483.72  5127.1  484.27  5298.6  489.95  5325.1  490.95
  5354.0  490.82  5381.6  491.40  5409.9  491.17  5424.0  493.52  5494.8  495.96
#Mann=10,-1,0
  4440.8    0.05       0  4461.9    0.07       0  4588.9    0.05       0
  4828.8    0.12       0  4835.3    0.12       0  4994.1    0.07       0
  4999.9    0.12       0  5028.1    0.07       0  5298.6   0.045       0
  5354.0    0.07       0
Bank Sta=4994.1,4999.9
Exp/Cntr=0.3,0.1

Type RM Length L Ch R = 1,20604,456,456,456
BEGIN DESCRIPTION:
SAUL CREEK 45.0
END DESCRIPTION:
XS GIS Cut Line= 3
      2322775.01     13753275.02      2322625.00     13752975.00
      2322625.00     13752325.03
#Sta/Elev= 30
  4660.0  491.70  4696.4  491.90  4713.1  490.45  4749.5  489.19  4808.2  489.60
  4847.3  487.21  4883.6  487.36  4892.0  486.34  4922.9  484.95  4959.1  483.03
  4981.5  478.37  5002.5  476.74  5003.0  476.24  5008.4  476.74  5025.4  477.45
  5035.4  480.92  5045.4  482.72  5055.4  483.31  5093.9  482.66  5115.4  481.56
  5195.4  483.56  5315.4  485.19  5335.4  486.26  5355.4  485.81  5423.7  488.08
  5485.4  489.22  5565.4  492.14  5585.4  492.28  5615.4  494.61  5645.4  494.19
#Mann=6,-1,0
  4660.0    0.05       0  4922.9    0.12       0  5002.5    0.07       0
  5008.4    0.12       0  5093.9    0.07       0  5423.7   0.045       0
Bank Sta=5002.5,5008.4
Exp/Cntr=0.3,0.1

Type RM Length L Ch R = 1,20148,475,475,475
BEGIN DESCRIPTION:
SAUL CREEK 44.0
END DESCRIPTION:
XS GIS Cut Line= 3
      2322824.99     13753275.04      2322975.00     13752775.00
      2322874.99     13752374.96
#Sta/Elev= 30
  4477.7  491.79  4550.8  489.32  4582.1  489.70  4631.7  487.09  4697.0  487.06
  4717.5  485.70  4728.3  485.43  4736.1  484.02  4741.4  485.02  4759.6  478.17
  4769.2  478.69  4774.4  477.79  4780.5  479.20  4801.4  480.00  4845.8  477.49
  4864.0  481.46  4878.8  481.93  4944.9  480.25  4950.2  481.06  4968.4  477.02
  4980.2  476.00  4980.7  475.50  4986.2  476.00  4997.1  478.56  5021.7  479.72
  5071.9  480.71  5082.2  479.86  5123.9  481.33  5226.1  484.98  5412.1  492.58
#Mann=7,-1,0
  4477.7    0.05       0  4717.5    0.07       0  4980.2    0.07       0
  4986.2    0.07       0  5021.7    0.12       0  5123.9    0.07       0
  5226.1   0.045       0
Bank Sta=4980.2,4986.2
Exp/Cntr=0.3,0.1

Type RM Length L Ch R = 1,19673,453,453,453
BEGIN DESCRIPTION:
SAUL CREEK 43.0
END DESCRIPTION:
XS GIS Cut Line= 3
      2323425.00     13753325.04      2323375.00     13752625.00
      2323275.02     13752325.05
#Sta/Elev= 30
  4298.1  490.37  4318.2  490.28  4365.8  488.15  4438.5  487.92  4458.5  486.55
  4498.6  486.08  4548.8  484.42  4679.1  482.93  4699.2  481.69  4735.5  480.65
  4786.9  479.10  4858.6  477.96  4919.7  478.72  4939.8  477.87  4957.5  478.11
  4979.9  476.19  5002.6  477.15  5007.5  474.93  5008.0  474.43  5013.0  474.43
  5013.5  474.93  5021.0  479.29  5031.5  480.54  5059.8  480.57  5115.9  483.15
  5137.0  483.02  5247.5  487.35  5269.4  489.21  5274.0  489.74  5316.1  489.81
#Mann=9,-1,0
  4298.1    0.05       0  4735.5    0.07       0  4858.6    0.12       0
  4957.5    0.12       0  5007.5    0.07       0  5013.5    0.12       0
  5059.8   0.045       0  5247.5    0.07       0  5269.4   0.045       0
Bank Sta=5007.5,5013.5
Exp/Cntr=0.3,0.1

Type RM Length L Ch R = 1,19220,468,468,468
BEGIN DESCRIPTION:
SAUL CREEK 42.0
END DESCRIPTION:
XS GIS Cut Line= 3
      2323725.00     13753174.97      2323775.00     13752775.00
      2323725.00     13752174.96
#Sta/Elev= 30
  4593.1  488.43  4613.2  488.48  4630.9  487.26  4693.8  485.46  4744.2  483.49
  4845.0  481.22  4877.8  481.28  4893.6  480.29  4915.6  478.42  4925.6  478.20
  4953.3  476.37  4965.9  476.03  4993.8  474.40  4998.7  474.40  5003.1  472.92
  5003.6  472.42  5008.8  472.42  5009.3  472.92  5021.0  473.10  5036.3  473.53
  5053.9  476.48  5066.4  477.35  5106.6  476.59  5126.6  476.63  5191.8  478.00
  5317.3  482.36  5327.3  482.29  5377.5  483.62  5389.9  484.38  5598.3  488.48
#Mann=8,-1,0
  4593.1    0.05       0  4893.6    0.07       0  4993.8    0.12       0
  5003.1    0.07       0  5009.3    0.12       0  5021.0   0.035       0
  5191.8   0.045       0  5389.9    0.07       0
Bank Sta=5003.1,5009.3
Exp/Cntr=0.3,0.1

Type RM Length L Ch R = 1,18752,454,454,454
BEGIN DESCRIPTION:
SAUL CREEK 41.0
END DESCRIPTION:
XS GIS Cut Line= 3
      2323925.00     13753124.99      2324025.00     13752625.00
      2324175.00     13752325.00
#Sta/Elev= 30
  4490.6  486.60  4531.4  485.78  4551.8  484.44  4592.6  484.32  4623.2  482.79
  4674.2  482.06  4755.7  478.66  4776.1  478.44  4796.5  477.19  4838.5  476.61
  4898.5  475.30  4938.3  475.68  4969.9  475.13  4980.1  474.19  4997.9  470.56
  5003.3  470.56  5011.3  469.54  5011.8  469.04  5017.1  469.04  5017.6  469.54
  5031.2  474.79  5036.8  474.16  5053.6  476.22  5059.2  475.76  5067.6  477.14
  5076.0  477.49  5132.9  478.77  5260.4  482.96  5282.8  484.73  5335.9  485.88
#Mann=6,-1,0
  4490.6   0.035       0  4838.5    0.07       0  4938.3    0.12       0
  5011.3    0.07       0  5017.6    0.12       0  5132.9    0.07       0
Bank Sta=5011.3,5017.6
Exp/Cntr=0.3,0.1

Type RM Length L Ch R = 1,18298,483,483,483
BEGIN DESCRIPTION:
SAUL CREEK 40.0
END DESCRIPTION:
XS GIS Cut Line= 3
      2324024.98     13753075.02      2324425.00     13752675.00
      2324425.00     13752375.02
#Sta/Elev= 30
  4434.4  484.74  4505.1  482.34  4533.4  482.18  4561.7  480.77  4590.0  480.82
  4632.4  479.58  4660.7  479.32  4703.1  477.71  4745.6  477.19  4759.7  476.61
  4802.1  476.55  4833.2  474.93  4858.7  474.98  4887.0  473.60  4957.7  473.58
  4968.4  472.78  4971.8  472.53  4986.0  469.85  4993.4  469.14  4993.9  468.64
  4999.3  468.64  4999.8  469.14  5010.1  469.67  5030.1  472.35  5040.1  472.71
  5090.1  476.51  5116.4  477.87  5150.1  478.85  5287.5  485.34  5300.1  486.53
#Mann=7,-1,0
  4434.4   0.035       0  4833.2    0.07       0  4968.4    0.12       0
  4993.4    0.07       0  4999.8    0.12       0  5116.4    0.07       0
  5287.5    0.05       0
Bank Sta=4993.4,4999.8
Exp/Cntr=0.3,0.1

Type RM Length L Ch R = 1,17815,481,481,481
BEGIN DESCRIPTION:
SAUL CREEK 39.0
END DESCRIPTION:
XS GIS Cut Line= 3
      2324875.00     13753125.04      2324875.00     13752775.00
      2324975.01     13752474.96
#Sta/Elev= 30
  4645.4  480.20  4735.4  478.02  4755.4  477.85  4815.4  474.92  4845.4  474.56
  4885.4  473.45  4915.4  473.63  4936.1  472.99  4955.4  472.43  4965.4  471.13
  4998.1  469.83  5006.0  468.28  5012.5  464.79  5013.0  464.29  5020.0  464.29
  5020.5  464.79  5027.1  465.66  5037.6  469.93  5048.1  472.01  5069.2  472.22
  5100.8  473.89  5128.1  473.91  5164.1  474.82  5185.2  475.75  5195.7  476.68
  5227.3  478.13  5237.9  479.14  5248.4  478.95  5290.6  480.71  5311.7  482.09
#Mann=5,-1,0
  4645.4    0.05       0  4936.1    0.12       0  5012.5    0.07       0
  5020.5    0.12       0  5128.1    0.07       0
Bank Sta=5012.5,5020.5
Exp/Cntr=0.3,0.1

Type RM Length L Ch R = 1,17334,449,449,449
BEGIN DESCRIPTION:
SAUL CREEK 38.0
END DESCRIPTION:
XS GIS Cut Line= 3
      2325275.01     13753074.97      2325325.00     13752775.00
      2325325.00     13752475.00
#Sta/Elev= 30
  4699.7  480.00  4709.8  479.45  4727.5  479.26  4750.4  477.75  4760.5  476.66
  4821.3  473.35  4841.6  471.95  4861.9  471.33  4882.1  470.28  4891.2  470.13
  4910.0  469.14  4915.1  468.43  4922.7  467.90  4970.9  465.13  4975.9  464.46
  4979.5  463.60  4980.0  463.10  4987.0  463.10  4987.5  463.60  4993.7  464.21
  5001.3  466.79  5006.3  466.79  5013.8  468.73  5023.8  470.78  5043.8  472.07
  5068.3  472.79  5113.8  473.81  5153.8  475.72  5183.8  476.22  5303.8  480.92
#Mann=5,-1,0
  4699.7    0.05       0  4891.2    0.12       0  4979.5    0.07       0
  4987.5    0.12       0  5068.3    0.05       0
Bank Sta=4979.5,4987.5
Exp/Cntr=0.3,0.1

Type RM Length L Ch R = 1,16885,467,467,467
BEGIN DESCRIPTION:
SAUL CREEK 37.0
END DESCRIPTION:
XS GIS Cut Line= 3
      2325624.99     13753175.04      2325675.00     13752875.00
      2325675.00     13752474.98
#Sta/Elev= 30
  4699.8  478.80  4721.9  478.46  4788.5  474.08  4793.6  474.33  4811.4  473.13
  4849.4  471.70  4854.4  471.09  4899.2  469.58  4915.3  468.34  4943.2  467.46
  4963.4  466.08  4976.1  464.84  4989.8  461.63  4990.3  461.13  4997.4  461.13
  4997.9  461.63  5006.5  462.13  5014.0  464.05  5024.0  467.51  5034.0  469.14
  5054.0  470.31  5072.2  469.74  5084.0  469.53  5114.0  471.08  5174.0  471.54
  5234.0  472.92  5274.0  475.20  5324.0  477.05  5354.0  478.90  5404.0  480.74
#Mann=6,-1,0
  4699.8   0.045       0  4721.9    0.05       0  4899.2    0.12       0
  4989.8    0.07       0  4997.9    0.12       0  5072.2    0.05       0
Bank Sta=4989.8,4997.9
Exp/Cntr=0.3,0.1

Type RM Length L Ch R = 1,16418,483,483,483
BEGIN DESCRIPTION:
SAUL CREEK 36.0
END DESCRIPTION:
XS GIS Cut Line= 3
      2326125.00     13753125.03      2326125.00     13752925.00
      2326125.00     13752525.03
#Sta/Elev= 30
  4795.4  476.50  4845.4  474.17  4865.4  472.61  4885.4  471.87  4925.4  468.39
  4945.4  467.24  4955.4  467.22  4972.5  466.45  4985.4  465.42  4992.9  463.27
  4997.9  463.27  5005.4  460.33  5011.3  459.82  5011.8  459.32  5019.0  459.32
  5019.5  459.82  5025.4  461.62  5035.4  463.78  5045.4  465.07  5075.4  464.34
  5085.4  465.30  5105.4  465.70  5115.4  466.70  5137.8  467.17  5175.4  468.33
  5205.4  468.65  5295.4  472.33  5325.4  474.15  5369.4  477.67  5395.4  479.41
#Mann=6,-1,0
  4795.4    0.05       0  4972.5    0.12       0  5011.3    0.07       0
  5019.5    0.12       0  5137.8    0.05       0  5369.4    0.07       0
Bank Sta=5011.3,5019.5
Exp/Cntr=0.3,0.1

Type RM Length L Ch R = 1,15935,473,473,473
BEGIN DESCRIPTION:
SAUL CREEK 35.0
END DESCRIPTION:
XS GIS Cut Line= 3
      2326575.00     13753125.02      2326575.00     13752925.00
      2326674.99     13752525.03
#Sta/Elev= 30
  4795.8  474.10  4855.8  471.99  4925.8  466.74  4945.8  465.84  4962.8  463.99
  4975.8  463.05  4998.4  462.98  5006.1  460.49  5014.8  459.39  5015.3  458.89
  5022.7  458.89  5023.2  459.39  5037.0  463.49  5060.2  463.12  5101.5  465.02
  5171.0  466.23  5183.9  466.62  5208.7  468.36  5220.0  469.44  5225.2  469.25
  5243.2  470.10  5253.5  471.56  5266.4  472.28  5302.5  478.45  5307.6  478.15
  5325.7  481.20  5376.3  486.03  5384.9  487.35  5390.1  487.20  5408.1  488.98
#Mann=6,-1,0
  4795.8    0.05       0  4962.8    0.07       0  5014.8    0.07       0
  5023.2    0.07       0  5208.7    0.12       0  5376.3    0.07       0
Bank Sta=5014.8,5023.2
Exp/Cntr=0.3,0.1

Type RM Length L Ch R = 1,15462,465,465,465
BEGIN DESCRIPTION:
SAUL CREEK 34.0
END DESCRIPTION:
XS GIS Cut Line= 3
      2326775.02     13753224.97      2327025.00     13752825.00
      2327025.00     13752724.97
#Sta/Elev= 30
  4539.0  480.35  4567.9  478.97  4583.2  476.45  4619.7  473.58  4662.2  472.33
  4698.8  469.28  4771.9  465.64  4841.3  463.46  4872.1  462.44  4929.9  462.54
  4939.3  461.11  4945.2  462.31  4951.7  460.92  4955.3  458.94  4960.5  456.07
  4966.4  460.04  4975.3  457.62  4977.6  456.01  4978.1  455.51  4985.5  455.51
  4986.0  456.01  4987.7  458.14  5003.0  456.33  5007.7  460.44  5013.2  460.44
  5020.7  462.91  5030.7  464.99  5050.7  467.89  5090.7  471.91  5110.7  475.21
#Mann=5,-1,0
  4539.0    0.05       0  4841.3    0.12       0  4955.3    0.07       0
  4977.6    0.07       0  4986.0    0.07       0
Bank Sta=4977.6,4986
Exp/Cntr=0.3,0.1

Type RM Length L Ch R = 1,14997,466,466,466
BEGIN DESCRIPTION:
SAUL CREEK 33.0
END DESCRIPTION:
XS GIS Cut Line= 3
      2327524.98     13753274.96      2327425.00     13753025.00
      2327325.01     13752625.02
#Sta/Elev= 30
  4725.4  477.87  4735.9  477.74  4764.4  476.34  4794.0  473.30  4818.3  470.07
  4847.9  468.56  4872.1  465.87  4926.0  461.95  4997.2  459.46  5012.7  455.66
  5017.8  457.28  5021.3  454.32  5021.8  453.82  5029.3  453.82  5029.8  454.32
  5038.2  457.10  5046.2  459.71  5095.1  460.22  5136.3  462.62  5141.5  462.33
  5200.8  465.83  5242.7  469.79  5283.2  476.55  5314.2  483.54  5334.8  487.37
  5347.7  490.75  5355.4  492.12  5370.0  493.17  5388.9  494.82  5406.9  495.38
#Mann=7,-1,0
  4725.4    0.07       0  4735.9    0.12       0  5021.3    0.07       0
  5029.8    0.12       0  5038.2    0.07       0  5242.7    0.12       0
  5370.0   0.035       0
Bank Sta=5021.3,5029.8
Exp/Cntr=0.3,0.1

Type RM Length L Ch R = 1,14531,447,447,447
BEGIN DESCRIPTION:
SAUL CREEK 32.0
END DESCRIPTION:
XS GIS Cut Line= 3
      2327825.01     13753124.96      2327875.00     13752975.00
      2327624.99     13752624.99
#Sta/Elev= 30
  4837.2  469.71  4932.0  460.17  4963.7  457.85  4974.2  455.02  4980.5  452.56
  4981.0  452.06  4988.5  452.06  4989.0  452.56  4998.3  453.23  5002.6  457.55
  5008.8  458.76  5025.3  458.17  5032.1  457.80  5094.8  458.96  5118.2  458.31
  5215.8  462.24  5246.0  463.31  5275.5  466.91  5281.6  466.50  5302.5  471.39
  5311.1  474.17  5317.2  474.02  5325.8  476.88  5332.0  476.79  5346.7  482.29
  5352.9  482.26  5361.5  484.57  5367.6  485.21  5388.5  489.87  5425.4  493.57
#Mann=5,-1,0
  4837.2    0.12       0  4980.5    0.07       0  4989.0    0.12       0
  5025.3    0.07       0  5215.8    0.12       0
Bank Sta=4980.5,4989
Exp/Cntr=0.3,0.1

Type RM Length L Ch R = 1,14084,442,442,442
BEGIN DESCRIPTION:
SAUL CREEK 31.0
END DESCRIPTION:
XS GIS Cut Line= 3
      2328125.01     13753374.97      2328275.00     13752825.00
      2327874.96     13752574.98
#Sta/Elev= 30
  4435.9  478.43  4487.7  476.64  4498.1  468.57  4514.2  464.19  4532.6  461.73
  4549.9  462.89  4622.4  457.37  4641.4  457.37  4681.2  462.18  4767.6  455.40
  4795.2  454.68  4809.0  456.24  4819.4  453.93  4829.7  454.84  4850.5  462.11
  4869.1  463.57  4933.4  457.76  4988.7  456.81  5003.4  452.34  5008.9  452.34
  5009.4  450.87  5009.9  450.37  5017.9  450.87  5019.5  454.14  5034.8  457.81
  5113.3  457.22  5187.0  456.84  5274.6  461.13  5360.3  464.86  5477.7  475.05
#Mann=7,-1,0
  4435.9   0.035       0  4514.2    0.07       0  4869.1    0.12       0
  5009.4    0.07       0  5017.9    0.12       0  5113.3    0.07       0
  5274.6    0.12       0
Bank Sta=5009.4,5017.9
Exp/Cntr=0.3,0.1

Type RM Length L Ch R = 1,13642,446,446,446
BEGIN DESCRIPTION:
SAUL CREEK 30.0
END DESCRIPTION:
XS GIS Cut Line= 3
      2328775.04     13752725.02      2328575.00     13752625.00
      2327775.00     13752375.00
#Sta/Elev= 30
  4780.7  466.94  4794.7  464.86  4892.5  461.21  4945.7  457.54  4968.0  454.42
  4973.6  452.58  4975.6  448.75  4976.1  448.25  4988.3  448.75  4996.0  449.71
  5001.6  452.55  5007.0  452.55  5014.8  456.28  5020.6  457.02  5090.8  455.96
  5361.1  456.23  5393.6  458.46  5425.0  463.01  5466.7  467.45  5475.8  469.19
  5485.8  468.80  5496.8  464.90  5580.6  466.24  5593.7  467.13  5612.0  470.55
  5658.6  471.98  5696.4  474.73  5723.6  479.04  5780.5  482.23  5842.5  485.80
#Mann=6,-1,0
  4780.7    0.12       0  4975.6    0.07       0  4988.3    0.12       0
  5425.0    0.12       0  5466.7    0.07       0  5780.5    0.12       0
Bank Sta=4975.6,4988.3
Exp/Cntr=0.3,0.1

Type RM Length L Ch R = 1,13196,436,436,436
BEGIN DESCRIPTION:
SAUL CREEK 29.0
END DESCRIPTION:
XS GIS Cut Line= 3
      2329274.98     13752524.99      2328525.00     13752325.00
      2328124.99     13752225.00
#Sta/Elev= 30
  4228.6  482.44  4235.3  482.23  4384.2  475.35  4481.5  468.75  4539.1  467.96
  4580.5  465.17  4596.6  462.03  4636.7  463.67  4735.7  459.92  4751.9  457.42
  4757.0  459.09  4808.1  458.06  4818.5  457.24  4826.9  449.38  4832.8  448.34
  4833.3  447.84  4845.5  448.34  4872.2  448.53  4880.6  453.68  4897.3  452.01
  4963.4  452.14  4999.6  449.26  5004.3  448.82  5015.1  448.39  5022.8  453.12
  5028.0  451.73  5046.0  455.83  5275.4  456.88  5357.8  461.65  5417.1  468.20
#Mann=8,-1,0
  4228.6    0.05       0  4235.3   0.035       0  4384.2    0.12       0
  4832.8    0.07       0  4845.5    0.12       0  4897.3    0.07       0
  4999.6    0.12       0  5004.3    0.07       0
Bank Sta=4832.8,4845.5
Exp/Cntr=0.3,0.1

Type RM Length L Ch R = 1,12760,415,415,415
BEGIN DESCRIPTION:
SAUL CREEK 28.0
END DESCRIPTION:
XS GIS Cut Line= 3
      2329175.00     13752125.00      2328725.00     13752025.00
      2327725.01     13751525.01
#Sta/Elev= 30
  4535.7  474.11  4576.7  472.21  4689.4  461.64  4846.6  456.10  4923.7  454.57
  4935.2  452.21  4939.1  448.48  4939.6  447.98  4951.9  448.48  4972.4  450.07
  4977.5  449.07  4994.1  452.06  5019.0  453.10  5153.2  454.02  5220.3  452.17
  5315.4  454.54  5452.3  458.43  5490.3  461.28  5502.6  462.76  5533.3  462.68
  5547.3  461.70  5564.1  457.27  5667.5  457.84  5698.2  458.88  5734.4  466.29
  5770.9  477.81  5836.0  482.88  5882.7  484.68  6033.7  494.48  6114.7  497.23
#Mann=8,-1,0
  4535.7    0.12       0  4846.6    0.12       0  4939.1    0.07       0
  4951.9    0.12       0  5315.4    0.12       0  5490.3    0.07       0
  5734.4    0.05       0  5836.0    0.07       0
Bank Sta=4939.1,4951.9
Exp/Cntr=0.3,0.1

Type RM Length L Ch R = 1,12345,429,429,429
BEGIN DESCRIPTION:
SAUL CREEK 27.0
END DESCRIPTION:
XS GIS Cut Line= 3
      2329174.97     13751924.99      2328575.00     13751725.00
      2328374.99     13751424.98
#Sta/Elev= 30
  4367.5  471.87  4420.2  468.63  4483.4  459.45  4515.0  457.02  4641.5  453.52
  4841.8  451.62  4871.0  452.55  4978.8  453.46  5002.9  451.17  5007.0  448.43
  5007.5  447.93  5019.9  448.43  5058.5  449.13  5064.5  451.36  5108.1  451.09
  5121.6  456.12  5130.6  456.57  5144.1  460.09  5157.7  461.82  5172.7  459.55
  5187.7  454.56  5193.7  456.08  5202.7  454.98  5225.1  457.68  5238.8  459.79
  5244.8  463.66  5259.8  467.03  5288.4  468.34  5310.9  471.73  5360.5  472.63
#Mann=5,-1,0
  4367.5    0.12       0  4871.0    0.12       0  5007.0    0.07       0
  5019.9    0.12       0  5225.1    0.07       0
Bank Sta=5007,5019.9
Exp/Cntr=0.3,0.1

Type RM Length L Ch R = 1,11916,473,473,473
BEGIN DESCRIPTION:
SAUL CREEK 26.0
END DESCRIPTION:
XS GIS Cut Line= 3
      2329275.03     13751575.01      2328825.00     13751425.00
      2328525.00     13751325.00
#Sta/Elev= 30
  4515.2  471.48  4557.4  468.57  4567.9  465.79  4594.3  462.91  4599.6  461.50
  4620.6  459.26  4631.2  457.23  4658.0  455.07  4694.4  453.18  4760.8  452.02
  4873.6  450.53  4905.2  449.03  4915.8  447.41  4926.3  449.33  4966.4  451.07
  4992.2  449.20  5000.1  446.72  5004.2  440.61  5004.7  440.11  5017.1  440.61
  5031.7  441.97  5042.3  449.60  5052.8  450.77  5105.5  452.03  5137.1  451.72
  5171.9  453.96  5189.9  455.40  5221.5  459.95  5247.7  461.60  5305.8  466.11
#Mann=8,-1,0
  4515.2    0.12       0  4658.0    0.12       0  4760.8    0.12       0
  4966.4    0.12       0  5004.2    0.07       0  5017.1    0.12       0
  5171.9    0.12       0  5247.7    0.07       0
Bank Sta=5004.2,5017.1
Exp/Cntr=0.3,0.1

Type RM Length L Ch R = 1,11443,478,478,478
BEGIN DESCRIPTION:
SAUL CREEK 25.0
END DESCRIPTION:
XS GIS Cut Line= 3
      2329374.98     13751274.99      2329025.00     13751125.00
      2328425.05     13751175.00
#Sta/Elev= 30
  4620.0  469.76  4652.6  468.19  4681.6  463.18  4728.8  458.98  4761.3  455.07
  4804.9  452.54  4864.9  450.92  4906.6  450.81  4915.5  450.95  4924.6  446.61
  4933.7  440.06  4950.7  439.84  4951.2  439.34  4963.7  439.84  4970.7  440.71
  4986.3  446.44  4991.7  444.10  4998.0  446.40  5003.3  446.40  5020.8  449.45
  5030.0  449.88  5081.0  448.71  5161.3  448.74  5271.7  450.10  5368.8  455.69
  5392.1  459.33  5419.7  462.37  5424.7  462.14  5540.1  469.78  5602.8  473.08
#Mann=9,-1,0
  4620.0    0.12       0  4761.3    0.12       0  4864.9    0.12       0
  4906.6    0.12       0  4950.7    0.07       0  4963.7    0.12       0
  4970.7    0.12       0  5030.0    0.12       0  5368.8    0.07       0
Bank Sta=4950.7,4963.7
Exp/Cntr=0.3,0.1

Type RM Length L Ch R = 1,10965,447,447,447
BEGIN DESCRIPTION:
SAUL CREEK 24.0
END DESCRIPTION:
XS GIS Cut Line= 3
      2329425.04     13750775.00      2328925.00     13750725.00
      2328725.03     13750625.02
#Sta/Elev= 30
  4492.9  469.12  4545.7  466.97  4553.2  465.77  4583.4  458.34  4603.5  455.32
  4623.6  452.41  4663.8  449.27  4704.0  447.90  4724.1  448.56  4764.3  447.83
  4834.6  448.51  4905.0  448.10  4925.1  447.77  4942.7  446.54  4954.1  447.86
  4965.3  447.44  4975.3  440.41  4978.9  440.07  4979.4  439.57  4991.9  440.07
  4992.9  441.06  5003.8  441.24  5009.4  443.01  5048.5  448.19  5058.5  448.46
  5098.8  448.55  5121.2  450.64  5130.8  452.30  5182.7  463.05  5219.0  466.85
#Mann=6,-1,0
  4492.9    0.12       0  4954.1    0.07       0  4978.9    0.07       0
  4991.9    0.07       0  5058.5    0.12       0  5130.8    0.07       0
Bank Sta=4978.9,4991.9
Exp/Cntr=0.3,0.1

Type RM Length L Ch R = 1,10518,464,464,464
BEGIN DESCRIPTION:
SAUL CREEK 23.0
END DESCRIPTION:
XS GIS Cut Line= 3
      2329375.03     13750475.01      2329175.00     13750375.00
      2328875.04     13750375.00
#Sta/Elev= 30
  4782.5  460.14  4818.9  457.27  4841.2  454.19  4858.0  449.69  4863.6  449.47
  4872.0  446.93  4882.3  445.72  4902.7  444.69  4930.7  446.07  4947.4  445.63
  4953.0  440.98  4961.4  435.97  4969.6  432.95  4985.5  432.51  4986.0  432.01
  4998.4  432.01  4998.9  432.51  5003.3  433.35  5008.6  433.35  5016.1  439.34
  5026.1  444.40  5036.1  445.75  5056.1  445.24  5076.1  447.12  5190.8  447.97
  5216.1  448.37  5236.1  450.12  5246.1  451.59  5286.1  460.66  5306.1  462.58
#Mann=6,-1,0
  4782.5    0.12       0  4882.3    0.12       0  4969.6    0.12       0
  4985.5    0.07       0  4998.9    0.12       0  5190.8    0.07       0
Bank Sta=4985.5,4998.9
Exp/Cntr=0.3,0.1

Type RM Length L Ch R = 1,10054,297,297,297
BEGIN DESCRIPTION:
SAUL CREEK 22.0
END DESCRIPTION:
XS GIS Cut Line= 3
      2329575.02     13750175.02      2329425.00     13750025.00
      2329024.98     13749975.00
#Sta/Elev= 30
  4784.1  462.27  4798.3  462.39  4829.2  461.01  4854.8  457.43  4897.3  449.31
  4911.4  447.30  4938.1  445.39  4982.1  445.06  4992.7  441.95  4998.8  441.95
  5009.7  431.28  5010.2  430.78  5022.6  430.78  5023.1  431.28  5026.5  437.91
  5034.1  442.05  5046.7  444.54  5056.7  445.04  5097.0  444.56  5114.7  443.92
  5119.7  442.62  5127.3  441.86  5218.0  445.81  5268.4  446.64  5292.6  448.93
  5328.8  454.76  5356.5  460.84  5361.6  460.75  5369.1  461.91  5399.4  463.61
#Mann=6,-1,0
  4784.1    0.07       0  4829.2    0.12       0  4938.1    0.12       0
  5009.7    0.07       0  5023.1    0.12       0  5292.6    0.07       0
Bank Sta=5009.7,5023.1
Exp/Cntr=0.3,0.1

Type RM Length L Ch R = 1,9757,150,150,150
BEGIN DESCRIPTION:
E20754
END DESCRIPTION:
XS GIS Cut Line= 3
      2329609.92     13750169.75      2329395.46     13749794.45
      2329014.83     13749617.53
#Sta/Elev= 30
  4537.3  462.54  4601.9  461.34  4649.8  455.45  4698.3  445.90  4748.0  444.61
  4816.4  445.47  4946.0  444.70  5006.3  435.38  5007.5  430.10  5008.0  429.60
  5020.9  430.10  5023.6  433.02  5074.9  445.37  5143.6  447.95  5172.0  454.64
  5189.4  456.19  5212.3  461.96  5217.8  464.31  5223.7  464.44  5234.7  461.74
  5240.7  458.98  5263.6  453.81  5269.1  456.35  5286.2  460.81  5292.0  464.25
  5309.3  465.61  5314.8  468.22  5322.9  469.28  5360.6  466.20  5389.3  466.65
#Mann=6,-1,0
  4537.3    0.07       0  4649.8    0.12       0  4748.0    0.12       0
  5007.5    0.07       0  5020.9    0.12       0  5286.2    0.07       0
Bank Sta=5007.5,5020.9
Exp/Cntr=0.3,0.1

Type RM Length L Ch R = 1,9607,434,434,434
BEGIN DESCRIPTION:
SAUL CREEK 21.0
END DESCRIPTION:
XS GIS Cut Line= 3
      2329625.00     13750125.01      2329475.00     13749675.00
      2329475.00     13749424.95
#Sta/Elev= 30
  4529.5  461.26  4582.2  458.61  4656.0  447.17  4666.5  447.17  4677.1  445.77
  4700.3  444.60  4740.3  445.22  4748.2  444.56  4887.9  444.23  4898.4  443.08
  4919.5  442.51  4961.7  442.63  4972.2  439.34  4982.8  432.50  4986.6  432.17
  4987.1  431.67  5000.1  432.17  5001.2  439.52  5013.9  439.76  5023.9  436.81
  5033.9  436.65  5053.9  440.82  5073.9  438.21  5093.9  444.59  5103.9  446.11
  5153.9  447.12  5173.9  448.49  5203.9  455.67  5223.9  459.52  5253.9  462.93
#Mann=5,-1,0
  4529.5    0.07       0  4700.3    0.12       0  4748.2    0.12       0
  4986.6    0.07       0  5000.1    0.12       0
Bank Sta=4986.6,5000.1
Exp/Cntr=0.3,0.1

Type RM Length L Ch R = 1,9173,260,260,260
BEGIN DESCRIPTION:
SAUL CREEK 20.0
END DESCRIPTION:
XS GIS Cut Line= 3
      2329925.00     13750125.04      2329875.00     13749675.00
      2329725.02     13749225.05
#Sta/Elev= 30
  4547.8  464.30  4568.0  462.71  4598.1  456.54  4654.9  450.84  4698.8  445.88
  4718.9  445.18  4940.2  444.06  4950.3  441.83  4960.4  435.91  4970.4  432.58
  4973.7  429.47  4974.2  428.97  4987.2  429.47  4998.1  430.45  5011.1  429.97
  5021.7  432.53  5032.2  438.08  5042.8  441.20  5063.9  442.15  5106.0  441.63
  5179.8  442.92  5316.8  441.38  5348.5  442.64  5359.0  443.89  5369.5  448.40
  5395.9  454.71  5401.2  457.46  5422.2  461.91  5443.3  463.80  5474.9  464.77
#Mann=4,-1,0
  4547.8    0.12       0  4654.9    0.12       0  4973.7    0.07       0
  4987.2    0.12       0
Bank Sta=4973.7,4987.2
Exp/Cntr=0.3,0.1

Type RM Length L Ch R = 1,8913,207,207,207
BEGIN DESCRIPTION:
E20752
END DESCRIPTION:
XS GIS Cut Line= 3
      2330510.55     13749955.25      2329953.02     13749413.81
      2329717.16     13749161.86
#Sta/Elev= 30
  4281.9  464.54  4406.2  463.54  4455.8  461.96  4533.5  462.65  4554.6  460.67
  4561.8  458.07  4568.8  457.81  4576.0  455.27  4604.3  450.93  4659.0  445.37
  4788.2  443.04  4950.7  443.20  4979.0  439.02  4986.2  432.83  4993.2  429.91
  4993.6  428.83  4994.1  428.33  5007.2  428.83  5007.3  432.35  5014.5  437.35
  5035.6  441.42  5078.1  440.48  5134.7  441.75  5212.4  440.38  5233.9  441.57
  5248.0  444.13  5290.3  458.60  5318.4  463.04  5335.0  464.12  5404.2  465.65
#Mann=5,-1,0
  4281.9    0.12       0  4659.0    0.12       0  4993.6    0.07       0
  5007.2    0.12       0  5335.0    0.12       0
Bank Sta=4993.6,5007.2
Exp/Cntr=0.3,0.1

Type RM Length L Ch R = 1,8706,256,256,256
BEGIN DESCRIPTION:
SAUL CREEK 19.0
END DESCRIPTION:
XS GIS Cut Line= 3
      2330424.98     13749474.99      2330075.00     13749275.00
      2329775.01     13749175.00
#Sta/Elev= 30
  4592.8  462.82  4615.8  461.31  4635.9  456.01  4650.4  452.32  4665.5  449.91
  4708.7  444.56  4767.7  441.98  4829.2  442.18  4982.2  441.72  4993.0  437.49
  4998.5  437.49  5006.4  430.84  5010.2  428.44  5010.7  427.94  5023.8  428.44
  5027.5  434.37  5038.0  438.08  5059.1  440.80  5090.8  440.22  5132.9  440.93
  5164.5  439.72  5185.6  441.58  5196.2  443.15  5206.7  447.15  5227.8  451.13
  5238.3  454.86  5259.4  458.49  5269.9  461.81  5286.6  463.43  5312.1  464.65
#Mann=6,-1,0
  4592.8    0.12       0  4635.9    0.12       0  4829.2    0.12       0
  5010.2    0.07       0  5023.8    0.12       0  5286.6    0.12       0
Bank Sta=5010.2,5023.8
Exp/Cntr=0.3,0.1

Type RM Length L Ch R = 1,8450,199,199,199
BEGIN DESCRIPTION:
E20753
END DESCRIPTION:
XS GIS Cut Line= 3
      2330633.92     13749263.71      2330070.97     13749033.17
      2329781.45     13749038.53
#Sta/Elev= 30
  4344.9  463.26  4397.6  462.59  4451.8  461.20  4473.4  459.64  4482.7  458.03
  4488.1  457.97  4505.8  453.19  4512.1  450.71  4517.5  450.76  4527.0  448.10
  4536.1  446.12  4565.5  443.06  4586.7  442.27  4678.7  440.79  4749.7  441.21
  4803.1  440.22  4880.5  440.89  4969.2  440.29  4989.2  438.75  4999.2  431.32
  5002.4  427.65  5002.9  427.15  5016.0  427.65  5019.2  428.07  5029.2  437.60
  5039.2  438.12  5059.2  443.10  5129.2  456.86  5189.2  461.85  5242.8  464.33
#Mann=6,-1,0
  4344.9    0.12       0  4397.6    0.12       0  4527.0    0.12       0
  4586.7    0.12       0  5002.4    0.07       0  5016.0    0.12       0
Bank Sta=5002.4,5016
Exp/Cntr=0.3,0.1
