--- BALDRIDGE CREEK.prj (project) ---

Proj Title=BALDRIDGE CREEK Base Level Engineering
Current Plan=p01
Default Exp/Contr=0.3,0.1
English Units
Geom File=g01
Flow File=f01
Plan File=p01
Y Axis Title=Elevation
X Axis Title(PF)=Main Channel Distance
X Axis Title(XS)=Station
BEGIN DESCRIPTION:
BALDRIDGE CREEK
END DESCRIPTION:
DSS Export Rating Curves= 0
DSS Export Rating Curve Sorted= 0
DSS Export Volume Flow Curves= 0
DXF OffsetX= 0
DXF OffsetY= 0
DXF ScaleX= 1
DXF ScaleY= 10

--- BALDRIDGE CREEK.p01 (plan) ---

Plan Title=Multiple Run
Program Version=4.10
Short Identifier=Multiple
Geom File=g01
Flow File=f01
Subcritical Flow
K Sum by GR= 0
Std Step Tol= 0.01
Critical Tol= 0.01
Num of Std Step Trials= 20
Max Error Tol= 0.3
Flow Tol Ratio= 0.001
Split Flow NTrial= 30
Split Flow Tol= 0.02
Split Flow Ratio= 0.02
Log Output Level= 0
Friction Slope Method= 1
Unsteady Friction Slope Method= 2
Unsteady Bridges Friction Slope Method= 1
Parabolic Critical Depth
Global Vel Dist= 1 , 1 , 1
Global Log Level= 0
CheckData=True
Encroach Param=-1 ,0,0, 0
BEGIN DESCRIPTION:
Multiple Run
END DESCRIPTION:
Computation Interval=1HOUR
Output Interval=1HOUR
Run HTab= 0
Run UNet= 0
Run PostProcess= 0
Run WQNet= 0
UNET Theta= 1
UNET Theta Warmup= 1
UNET ZTol= 0.02
UNET ZSATol= 0.05
UNET MxIter= 20
UNET MaxInSteps= 0
UNET DtIC= 0
UNET DtMin= 0
UNET MaxCRTS= 20
UNET WFStab= 2
UNET SFStab= 1
UNET WFX= 1
UNET SFX= 1
UNET DSS MLevel= 4
UNET DZMax Abort= 100
UNET Convert EG Bridges= 0
UNET Use Existing IB Tables=-1
UNET Froude Reduction=False
UNET Froude Limit= 1
UNET Froude Power= 10
UNET Time Slicing=0,0, 5
UNET Junction Losses=0
Instantaneous Interval=1HOUR
Write IC File= 0
Write IC File at Sim End=0
Echo Input=False
Echo Parameters=False
Echo Output=False
Write Detailed= 0
WQ AD Non Conservative
WQ ULTIMATE=-1
WQ Max Comp Step=1HOUR
WQ Output Interval=15MIN
WQ Output Selected Increments= 0
WQ Output face flow=0
WQ Output face velocity=0
WQ Output face area=0
WQ Output face dispersion=0
WQ Output cell volume=0
WQ Output cell surface area=0
WQ Output cell continuity=0
WQ Output cumulative cell continuity=0
WQ Output face conc=0
WQ Output face dconc_dx=0
WQ Output face courant=0
WQ Output face peclet=0
WQ Output face adv mass=0
WQ Output face disp mass=0
WQ Output cell mass=0
WQ Output cell source sink temp=0
WQ Output cell source sink nsm=0
WQ Output MaxMinRange=-1
WQ Daily Max Min Mean=-1
WQ Daily Range=0
WQ Daily Time=0
WQ Create Restart=0
WQ Fixed Restart=0
WQ System Summary=0
WQ Use Fixed Temperature=0
Sorting and Armoring Iterations= 10
XS Update Threshold= 0.02
Hydraulics Update Threshold= 0.02
Energy Slope Method= 1
Volume Change Method= 0
XS Weighting Method= 0
Number of US Weighted Cross Sections= 1
Number of DS Weighted Cross Sections= 1
Upstream XS Weight=0.25
Main XS Weight=0.5
Downstream XS Weight=0.25
Number of DS XS's Weighted with US Boundary= 1
Upstream Boundary Weight= 1
Weight of XSs Associated with US Boundary= 0
Number of US XS's Weighted with DS Boundary= 1
Downstream Boundary Weight= 0.5
Weight of XSs Associated with DS Boundary= 0.5
Sediment Output Level= 4
Mass or Volume Output= 0
Output Increment Type= 1
Profile and TS Output Increment= 10
XS Output Flag= 0
XS Output Increment= 10
Disregard all LS=0
Disregard all Conn=0
Disregard all Breaches=0
Disregard all Pumps=0

--- BALDRIDGE CREEK.f01 (steady flow) ---

Flow Title=Multiple
Number of Profiles=7
Profile Names=10-year,25-year,50-year,1pct_min,100-year,1pct_plu,500-year
River Rch & RM= BALDRIDGE CREEK,Reach-1,81430
     714    1150    1545    1005    2006    4002    3346
River Rch & RM= BALDRIDGE CREEK,Reach-1,77397
    1037    1708    2329    1536    3064    6114    5253
River Rch & RM= BALDRIDGE CREEK,Reach-1,76424
    1117    1831    2486    1631    3254    6492    5521
River Rch & RM= BALDRIDGE CREEK,Reach-1,70589
    1376    2271    3098    2039    4069    8119    6956
River Rch & RM= BALDRIDGE CREEK,Reach-1,67195
    1504    2484    3388    2230    4449    8877    7599
River Rch & RM= BALDRIDGE CREEK,Reach-1,60817
    1932    3226    4434    2938    5863   11697   10154
River Rch & RM= BALDRIDGE CREEK,Reach-1,58846
    2071    3459    4755    3150    6284   12539   10877
River Rch & RM= BALDRIDGE CREEK,Reach-1,53483
    2019    3362    4610    3046    6078   12127   10468
River Rch & RM= BALDRIDGE CREEK,Reach-1,49765
    2092    3480    4769    3148    6281   12531   10795
River Rch & RM= BALDRIDGE CREEK,Reach-1,41014
    2935    4941    6827    4539    9056   18069   15791
River Rch & RM= BALDRIDGE CREEK,Reach-1,33453
    2975    5006    6913    4594    9166   18289   15968
River Rch & RM= BALDRIDGE CREEK,Reach-1,30142
    3310    5583    7722    5138   10251   20454   17899
River Rch & RM= BALDRIDGE CREEK,Reach-1,26335
    3405    5742    7942    5283   10541   21031   18396
River Rch & RM= BALDRIDGE CREEK,Reach-1,19935
    3499    5901    8160    5427   10828   21605   18888
River Rch & RM= BALDRIDGE CREEK,Reach-1,14882
    3583    6040    8352    5553   11080   22107   19319
River Rch & RM= BALDRIDGE CREEK,Reach-1,10882
    3623    6106    8441    5611   11195   22336   19507
River Rch & RM= BALDRIDGE CREEK,Reach-1,7745
    3783    6374    8808    5852   11675   23295   20322
Boundary for River Rch & Prof#=BALDRIDGE CREEK,Reach-1,1
Up Type=0
Dn Type=3
Dn Slope=0.0001
Boundary for River Rch & Prof#=BALDRIDGE CREEK,Reach-1,2
Up Type=0
Dn Type=3
Dn Slope=0.0001
Boundary for River Rch & Prof#=BALDRIDGE CREEK,Reach-1,3
Up Type=0
Dn Type=3
Dn Slope=0.0001
Boundary for River Rch & Prof#=BALDRIDGE CREEK,Reach-1,4
Up Type=0
Dn Type=3
Dn Slope=0.0001
Boundary for River Rch & Prof#=BALDRIDGE CREEK,Reach-1,5
Up Type=0
Dn Type=3
Dn Slope=0.0001
Boundary for River Rch & Prof#=BALDRIDGE CREEK,Reach-1,6
Up Type=0
Dn Type=3
Dn Slope=0.0001
Boundary for River Rch & Prof#=BALDRIDGE CREEK,Reach-1,7
Up Type=0
Dn Type=3
Dn Slope=0.0001

--- BALDRIDGE CREEK.g01 (geometry) ---

Geom Title=Existing Conditions
Program Version=4.10

River Reach=BALDRIDGE CREEK ,Reach-1
Reach XY= 30
        2500325.       13816025.      2500227.04     13812980.85
      2501538.16     13810711.27      2502585.64     13810025.65
      2505023.84     13810221.88      2506416.05     13808631.68
      2505824.36     13805249.62      2506601.54      13802947.7
      2511085.16     13800264.72      2511476.46     13799028.54
      2513073.78     13798971.63       2513074.9     13798332.31
      2515319.55     13799172.96      2515772.26     13797980.34
      2516928.42     13798367.24      2519716.86     13796831.06
      2518925.36     13795559.73      2519278.49     13793876.27
      2520215.89     13793481.73       2519915.2     13792735.48
      2521020.03     13792577.58      2521491.64     13790308.32
      2522566.17       13790332.      2522024.96     13788044.76
      2522821.54     13787573.51      2522882.67     13785768.48
      2523935.18     13785814.68      2526321.55     13783223.75
      2527526.96     13775380.65        2528125.       13775475.

Type RM Length L Ch R = 1 ,81430   ,584,584,584
BEGIN DESCRIPTION:
BALDRIDGE CREEK 87.0
END DESCRIPTION:
XS GIS Cut Line= 3
      2500674.96     13816074.99      2500329.05     13815984.92
      2499825.04     13815875.01
#Sta/Elev= 30
  4637.9  427.49  4736.5  425.13  4777.1  424.79  4836.8  423.47  4906.5  422.16
  4937.5  422.18  4958.2  421.06  4968.5  421.97  4974.4  421.64  4979.6  421.04
  4987.2     417  4987.4   416.5  4990.9   416.5  4991.2     417  4994.8  419.41
    5000  419.41  5009.7  422.42  5030.2  421.83  5096.9  421.92  5109.6  422.19
  5114.7  421.43  5142.8  421.76  5183.7  421.47  5286.1  424.03  5316.8  424.02
  5378.2  425.89  5419.1  425.53  5449.8  426.92  5460.1  426.63  5511.2  427.77
#Mann= 6 ,-1 , 0
  4637.9     .05       0  4836.8     .07       0  4937.5     .12       0
  4987.2     .05       0  4991.2     .12       0  5096.9     .07       0
Bank Sta=4987.2,4991.2
XS Rating Curve= 0 ,0
Exp/Cntr=0.3,0.1

Type RM Length L Ch R = 1 ,80846   ,341,341,341
BEGIN DESCRIPTION:
BALDRIDGE CREEK 86.0
END DESCRIPTION:
XS GIS Cut Line= 3
      2500825.01       13815475.        2500525.       13815475.
      2499974.97     13815725.02
#Sta/Elev= 30
  4700.1  426.63  4730.1  426.29  4810.1  422.57  4900.1  420.13  4910.1  419.51
  4940.1  419.41  4950.1  419.85  4960.1  419.38  4973.8  416.77  4980.1  415.45
  4990.1     415  4995.6  414.26  4995.9  413.76  4999.4  413.76  4999.6  414.26
  5008.9  414.43  5014.4  417.47  5022.1  419.51  5037.5  419.79  5118.5  419.24
  5158.3  418.98  5204.4  419.49  5219.8  419.12  5279.1  419.96  5296.7  419.75
  5318.7  420.75  5362.6   420.7  5446.1  422.75  5474.6  422.65  5604.3  424.73
#Mann= 5 ,-1 , 0
  4700.1     .07       0  4973.8     .12       0  4995.6     .05       0
  4999.6     .12       0  5118.5     .07       0
Bank Sta=4995.6,4999.6
XS Rating Curve= 0 ,0
Exp/Cntr=0.3,0.1

Type RM Length L Ch R = 1 ,80505   ,552,552,552
BEGIN DESCRIPTION:
BALDRIDGE CREEK 85.0
END DESCRIPTION:
XS GIS Cut Line= 3
      2500975.04     13815325.01      2500447.01     13815241.27
      2499600.83      13815354.1
#Sta/Elev= 30
  4370.3  433.04  4489.4  427.15  4704.5  418.67  4775.3  417.41  4876.6  417.42
  4903.4  416.57  4987.7   417.5  5005.8  413.69  5006.1  413.19  5009.8  413.69
    5028  417.11  5058.3  418.53  5098.6  418.31  5108.7  416.74    5118  416.71
  5123.1     418    5139  418.93  5178.1  417.98  5209.6  418.54  5229.8  416.96
  5239.9  419.85  5330.8  420.56  5411.8  420.86  5431.6  421.02  5451.7  422.63
  5511.6  422.52  5562.7  423.78  5613.2  424.02  5673.7  425.82  5758.6  426.97
#Mann= 9 ,-1 , 0
  4370.3     .07       0  4489.4     .12       0  5005.8     .05       0
  5009.8     .12       0  5178.1     .07       0  5330.8     .12       0
  5411.8     .07       0  5511.6     .12       0  5562.7    .035       0
Bank Sta=5005.8,5009.8
XS Rating Curve= 0 ,0
Exp/Cntr=0.3,0.1

Type RM Length L Ch R = 1 ,79953   ,446,446,446
BEGIN DESCRIPTION:
BALDRIDGE CREEK 84.0
END DESCRIPTION:
XS GIS Cut Line= 3
      2500875.04     13814975.01        2500575.       13814925.
      2499675.03     13815274.99
#Sta/Elev= 30
  4695.8  425.69  4784.5  421.65  4817.5  421.37  4845.4  419.32    4858  419.54
  4898.6  417.03  4959.4  414.74  4979.7  414.79  4987.8  411.93  4988.1  411.43
  4991.8  411.93  4997.4  414.37  5009.6  415.12  5053.6  414.73    5064  413.73
  5096.5  415.79  5225.3   416.3  5407.7     419  5425.7  418.43  5431.1  417.18
  5461.3     419    5510   418.5  5569.2  419.51  5587.5  419.47  5672.2  420.23
  5718.9  421.25    5751   420.6  5840.6  421.99  5885.9  422.96  5965.6  424.89
#Mann= 9 ,-1 , 0
  4695.8     .12       0  4987.8     .05       0  4991.8     .12       0
  5096.5     .07       0  5569.2     .05       0  5587.5     .07       0
  5672.2    .035       0  5840.6     .12       0  5885.9    .035       0
Bank Sta=4987.8,4991.8
XS Rating Curve= 0 ,0
Exp/Cntr=0.3,0.1

Type RM Length L Ch R = 1 ,79507   ,455,455,455
BEGIN DESCRIPTION:
BALDRIDGE CREEK 83.0
END DESCRIPTION:
XS GIS Cut Line= 3
      2501190.66     13814605.32        2500425.       13814575.
      2499595.64     13814543.78
#Sta/Elev= 30
  4233.7  427.95  4277.9  427.48  4366.3  425.96  4429.5  423.74  4509.6  422.89
  4529.6   419.3  4549.1  418.73  4559.6  417.83  4589.6  417.94  4609.7  420.18
  4622.8  418.87  4639.7  419.65  4719.7  416.03  4739.8   416.3  4859.8  412.64
  4879.9  414.39  4989.9  413.22    5030  411.39    5050  412.33  5065.6  411.91
    5078  411.11  5078.3  410.61    5082  411.11    5120  412.87    5134  412.47
  5164.1  415.45  5390.2  416.35    5532  417.99  5754.9  421.98  5829.9  423.92
#Mann= 9 ,-1 , 0
  4233.7     .12       0  4277.9     .07       0  4549.1     .12       0
  5065.6     .07       0    5078     .05       0    5082     .07       0
  5164.1     .05       0    5532     .07       0  5754.9    .035       0
Bank Sta=5078,5082
XS Rating Curve= 0 ,0
Exp/Cntr=0.3,0.1

Type RM Length L Ch R = 1 ,79052   ,352,352,352
BEGIN DESCRIPTION:
BALDRIDGE CREEK 82.0
END DESCRIPTION:
XS GIS Cut Line= 3
      2501277.84     13814374.53        2500375.       13814175.
      2499841.84     13814061.69
#Sta/Elev= 30
  4079.3  426.24  4092.5  426.75  4098.9  424.14  4106.1  424.27  4112.9  424.74
  4376.2  418.09  4507.2  415.94  4607.4  414.05  4676.2  412.61  4696.7  413.54
  4768.4  411.88  4793.5  412.41    4922  409.18  4984.7  410.16  4993.7  408.28
  4999.4  405.34  4999.6  404.84  5003.4  405.34  5006.5  405.34  5014.2  410.06
  5044.8  409.92  5095.9  413.13  5163.4  413.77  5222.1  414.86  5271.7  414.06
  5310.6  415.12  5321.3  414.47  5364.7  415.03  5484.4   418.4    5549  419.09
#Mann= 8 ,-1 , 0
  4079.3     .05       0  4106.1    .035       0  4507.2     .05       0
  4607.4     .07       0  4793.5      .1       0  4999.4     .05       0
  5003.4      .1       0  5163.4     .07       0
Bank Sta=4999.4,5003.4
XS Rating Curve= 0 ,0
Exp/Cntr=0.3,0.1

Type RM Length L Ch R = 1 ,78700   ,467,467,467
BEGIN DESCRIPTION:
BALDRIDGE CREEK 81.0
END DESCRIPTION:
XS GIS Cut Line= 3
        2501242.     13813964.24      2500636.77     13813948.86
      2499934.18     13813887.32
#Sta/Elev= 30
  4383.3   420.8  4400.3  419.45  4792.7  412.54  4850.4  411.82  4870.5   412.2
    4953  410.89  4980.5  410.41  4992.1  409.52  5010.6  406.84  5018.6  403.88
  5018.9  403.38  5022.4  403.38  5022.6  403.88  5030.7  407.38  5040.7   408.4
  5070.8  408.44  5088.1  407.17    5111  407.34  5191.3  409.78  5248.8   410.1
  5291.6  412.28  5331.8  411.48  5402.1  412.74  5553.2  413.32  5592.8  414.33
  5612.9  415.69  5622.9  414.82    5653  415.84    5676  415.64    5694  415.99
#Mann= 7 ,-1 , 0
  4383.3     .05       0  4792.7    .035       0    4953      .1       0
  5018.6     .05       0  5022.6      .1       0  5248.8    .035       0
    5676     .07       0
Bank Sta=5018.6,5022.6
XS Rating Curve= 0 ,0
Exp/Cntr=0.3,0.1

Type RM Length L Ch R = 1 ,78233   ,485,485,485
BEGIN DESCRIPTION:
BALDRIDGE CREEK 80.0
END DESCRIPTION:
XS GIS Cut Line= 3
        2501025.       13813625.      2500539.33     13813533.44
      2500075.02     13813724.99
#Sta/Elev= 30
    4464  414.12    4637  410.97  4657.7  411.24    4705  410.16  4710.1   410.8
  4718.4  409.75  4783.6  409.27  4811.5  409.02  4891.4  409.12  4911.2   408.3
  4942.3  406.48  4963.3  406.69  4971.9  404.75  4975.3  404.65  4975.5  404.15
    4979  404.15  4979.3  404.65  4984.5  406.28  5006.6  406.97  5049.1  406.81
  5071.1  405.81    5123  408.13  5168.4  408.59  5222.5  410.74  5262.1  411.06
  5277.5  410.54  5392.6  412.25  5406.4  413.32  5421.9  412.47  5460.5  413.35
#Mann= 8 ,-1 , 0
    4464     .05       0  4783.6     .07       0  4811.5     .05       0
  4911.2      .1       0  4975.3     .05       0  4979.3      .1       0
    5123     .07       0  5277.5    .035       0
Bank Sta=4975.3,4979.3
XS Rating Curve= 0 ,0
Exp/Cntr=0.3,0.1

Type RM Length L Ch R = 1 ,77748   ,351,351,351
BEGIN DESCRIPTION:
BALDRIDGE CREEK 79.0
END DESCRIPTION:
XS GIS Cut Line= 3
        2500975.       13813525.        2500375.       13813175.
        2500025.       13813475.
#Sta/Elev= 30
  4301.8  412.75  4413.2  411.05  4571.8   408.8  4744.9  407.58  4828.1  407.46
    4857  406.86  4871.1  406.14  4908.4  406.43  4915.4  405.67  4967.1  405.97
  4982.8  404.37  4988.6  404.93  4993.5  403.81  4999.7  403.81  5001.6  401.39
  5001.8  400.89  5005.3  400.89  5005.6  401.39  5024.4  404.47  5081.5  405.91
  5095.8  405.23  5102.3  405.89    5110  405.05  5116.6  405.16  5183.4  408.71
  5223.1  409.52  5280.1  409.28  5363.1  410.94  5400.9  410.95  5457.4  412.16
#Mann= 8 ,-1 , 0
  4301.8     .05       0  4413.2     .07       0  4744.9     .05       0
    4857      .1       0  5001.6     .05       0  5005.6      .1       0
  5183.4     .07       0  5363.1    .035       0
Bank Sta=5001.6,5005.6
XS Rating Curve= 0 ,0
Exp/Cntr=0.3,0.1

Type RM Length L Ch R = 1 ,77397   ,503,503,503
BEGIN DESCRIPTION:
X18096
END DESCRIPTION:
XS GIS Cut Line= 3
      2501082.99     13813241.12       2500354.7     13813000.06
      2499641.84      13812610.3
#Sta/Elev= 30
  4118.2  413.95  4190.2     410  4216.7  411.09  4421.7  408.75  4604.8  407.58
  4731.3  406.02  4832.4  403.74  4940.8  403.74  5007.6  403.81  5013.3   401.2
  5019.8  400.68    5020  400.18  5023.8  400.68  5035.1  403.87  5051.3  404.45
  5107.6  404.79  5147.1  404.23  5169.9  402.46  5176.5   404.1  5214.4  404.82
  5220.1   401.7  5236.2  404.04    5258  405.03  5263.7  406.44  5272.5  406.17
  5329.5  410.18    5376  411.38  5580.2  419.39  5604.1   419.5  5697.8  422.86
#Mann= 11 ,-1 , 0
  4118.2     .05       0  4421.7     .07       0  4604.8    .035       0
  4731.3      .1       0  4940.8     .07       0  5019.8     .05       0
  5023.8     .07       0  5051.3     .12       0  5107.6      .1       0
    5376     .12       0  5604.1     .05       0
Bank Sta=5019.8,5023.8
XS Rating Curve= 0 ,0
Exp/Cntr=0.3,0.1

Type RM Length L Ch R = 1 ,76894   ,470,470,470
BEGIN DESCRIPTION:
BALDRIDGE CREEK 78.0
END DESCRIPTION:
XS GIS Cut Line= 3
      2501274.98     13813174.99        2500475.       13812675.
      2500074.98     13812374.99
#Sta/Elev= 30
    4061  422.72    4163  415.55  4263.2  411.98  4561.6  405.93  4576.9  406.82
  4619.4  405.34  4634.7  407.55  4656.8  406.87    4686  405.55    4729  406.62
  4815.7   405.9  4838.7   405.1  4847.9  403.17  4859.9  401.74  4874.7  404.16
    4933  403.97  4954.3  399.76  4960.2  401.14    4969  399.35  4975.5   402.1
  4988.2  397.32  4988.6  396.82  4993.5  397.32  4996.7  399.59  5017.9  401.83
  5051.2  402.04  5067.9  401.32  5217.9  404.95  5337.4  410.32  5504.4  417.51
#Mann= 7 ,-1 , 0
    4061     .05       0  4656.8     .07       0  4847.9     .12       0
  4988.2     .05       0  4993.5     .12       0  5051.2      .1       0
  5337.4     .12       0
Bank Sta=4988.2,4993.5
XS Rating Curve= 0 ,0
Exp/Cntr=0.3,0.1

Type RM Length L Ch R = 1 ,76424   ,462,462,462
BEGIN DESCRIPTION:
BALDRIDGE CREEK 77.0
END DESCRIPTION:
XS GIS Cut Line= 3
      2501375.02     13813025.02        2500575.       13812275.
      2500374.97     13812074.97
#Sta/Elev= 30
  3902.9  420.65    3910   421.1    3931  418.88  4009.2  416.63  4037.5  414.74
    4080  415.05    4101  413.43  4242.6  410.21    4292  410.13  4341.6  408.46
  4511.3  405.91    4814  403.32  4879.1  400.94  4899.3  401.05  4971.4  401.66
  4978.3  400.49  4992.4  400.88  4996.1   399.9  5003.1   399.9    5011  397.29
  5011.4  396.79  5016.3  397.29  5027.8  399.83    5054   401.3  5084.4  403.86
  5112.7  403.89  5169.2  408.15  5206.7  409.54    5233  410.93  5282.4   413.3
#Mann= 8 ,-1 , 0
  3902.9     .05       0    4814     .07       0  4899.3     .12       0
    5011     .05       0  5016.3     .12       0    5054     .07       0
  5206.7      .1       0    5233     .12       0
Bank Sta=5011,5016.3
XS Rating Curve= 0 ,0
Exp/Cntr=0.3,0.1

Type RM Length L Ch R = 1 ,75962   ,483,483,483
BEGIN DESCRIPTION:
BALDRIDGE CREEK 76.0
END DESCRIPTION:
XS GIS Cut Line= 3
       2501626.6     13812820.56        2500925.       13812025.
       2500303.4     13811692.25
#Sta/Elev= 30
  3933.3  419.56  3944.8  419.29  4427.2  407.65  4582.8  407.08  4660.7  402.52
  4739.3  403.09  4788.7  409.76    4838  402.02  4874.1  400.37  4909.1  398.54
  4944.2  400.75  4995.3  397.99  4999.5   395.7  4999.9   395.2  5004.8   395.7
  5062.1  398.66    5068  400.97  5073.7  398.99  5084.2  400.86  5116.5  400.74
  5150.1  403.45  5155.7  406.51    5172  408.49  5177.7  411.53  5193.9  410.95
  5221.5  404.48  5325.6  404.73  5436.4   413.1  5682.9  419.78  5699.1   419.9
#Mann= 8 ,-1 , 0
  3933.3     .07       0  3944.8     .05       0  4874.1     .07       0
  4995.3     .12       0  4999.5     .05       0  5004.8     .12       0
  5116.5     .07       0  5682.9     .12       0
Bank Sta=4999.5,5004.8
XS Rating Curve= 0 ,0
Exp/Cntr=0.3,0.1

Type RM Length L Ch R = 1 ,75479   ,709,709,709
BEGIN DESCRIPTION:
X18095
END DESCRIPTION:
XS GIS Cut Line= 3
      2501852.27     13812756.18      2501323.48     13811785.14
      2500391.16     13811419.89
#Sta/Elev= 30
  3771.6  420.24  4012.1  414.58  4034.8  415.22  4066.2  413.28  4240.9  410.87
  4398.6  406.41  4478.9  405.85  4507.8  404.62  4902.9  401.31  4940.1  401.33
  4970.3  399.06  5000.1  398.67  5005.5  398.12  5015.3  395.32  5021.8  394.93
  5022.3  394.43  5027.2  394.93  5029.9  398.74  5036.8  399.31  5085.3   398.4
  5469.4  405.43  5541.5  408.43  5584.5  408.98  5656.6  412.35  5681.1  412.08
  5710.9  413.81  5746.1   413.3  5765.2  414.48  5819.4  415.29  5878.6  415.16
#Mann= 5 ,-1 , 0
  3771.6     .05       0  4902.9     .07       0  5021.8     .05       0
  5027.2     .07       0  5085.3     .05       0
Bank Sta=5021.8,5027.2
XS Rating Curve= 0 ,0
Exp/Cntr=0.3,0.1

Type RM Length L Ch R = 1 ,74770   ,792,792,792
BEGIN DESCRIPTION:
X18094
END DESCRIPTION:
XS GIS Cut Line= 3
      2502217.67     13812419.74      2501583.08     13811429.39
      2500371.66     13810660.23
#Sta/Elev= 30
  3415.8  414.25  3544.8  411.49  3680.5   407.9  3949.5   404.1  3955.9  404.99
  4131.2  403.33  4303.7  403.44  4808.6  398.03    4957  397.42  4969.4  396.56
  4978.7  393.81  4989.7  392.68  4990.2  392.18  4995.2  392.68  5005.8  397.04
    5021  397.98  5051.5  399.14  5078.6  398.56  5087.3  397.16  5093.9  394.21
  5099.8  394.65  5115.1  399.24  5185.8  401.35  5297.2  402.37  5388.3  405.81
  5609.5  411.64    5632  412.58  5750.4  415.46  5861.3  418.41    6027  420.75
#Mann= 11 ,-1 , 0
  3415.8     .05       0  3544.8     .07       0  3680.5     .05       0
  4808.6      .1       0  4989.7     .05       0  4995.2      .1       0
  5185.8     .07       0  5388.3     .05       0  5609.5     .07       0
    5632     .05       0  5750.4     .07       0
Bank Sta=4989.7,4995.2
XS Rating Curve= 0 ,0
Exp/Cntr=0.3,0.1

Type RM Length L Ch R = 1 ,73978   ,682,682,682
BEGIN DESCRIPTION:
BALDRIDGE CREEK 75.0
END DESCRIPTION:
XS GIS Cut Line= 3
      2502294.55     13812285.06       2501727.3     13810862.13
      2500910.06     13810131.42
#Sta/Elev= 30
  3226.8  411.67  3248.4  411.99  3360.6  407.59  3478.2  405.43  3882.7     402
  4187.3  400.69  4217.3  401.63  4524.6  399.66  4615.2  399.84  4658.6  399.32
    4734  396.27  4807.7  395.09  4815.2  395.83  4899.7  395.27  4963.2  396.38
  4977.5  395.47    4985  393.38  4988.7  391.09  4989.2  390.59  4994.7  391.09
  5013.4   397.4  5020.1  398.67  5062.7  400.61  5155.2  402.46  5296.8   406.2
  5331.9  408.22  5489.3  413.58  5572.6   417.8  5820.9  424.47  5854.9  425.59
#Mann= 10 ,-1 , 0
  3226.8     .05       0  3360.6     .07       0  3478.2     .05       0
  4524.6     .07       0  4615.2      .1       0  4988.7     .05       0
  4994.7      .1       0  5155.2     .05       0  5489.3     .07       0
  5820.9     .05       0
Bank Sta=4988.7,4994.7
XS Rating Curve= 0 ,0
Exp/Cntr=0.3,0.1

Type RM Length L Ch R = 1 ,73296   ,709,709,709
BEGIN DESCRIPTION:
BALDRIDGE CREEK 74.0
END DESCRIPTION:
XS GIS Cut Line= 3
      2502544.56     13811823.62        2502125.       13810775.
      2501611.94     13809814.14
#Sta/Elev= 30
  3871.2  403.23  4117.4   400.6  4623.7  398.47  4668.1  397.61    4687  394.51
  4799.6  394.31  4817.5  394.58  4824.3  397.78  4829.7  398.15  4848.5  403.57
  4860.6  405.75  4871.4   405.3  4907.8  397.46  4959.8   395.3  4991.2  393.38
    4998  391.31  5003.5  391.31  5005.7  388.49  5006.2  387.99  5011.9  388.49
  5014.5  391.27  5023.3  393.98  5030.7  394.58  5120.9  393.85  5370.6  397.79
  5503.7  401.43  5716.2  407.41  5732.5     409  5851.9  414.05  6089.9  425.48
#Mann= 8 ,-1 , 0
  3871.2     .05       0  4799.6     .12       0  4959.8      .1       0
  5005.7     .05       0  5011.9      .1       0  5120.9     .05       0
  5503.7     .07       0  5851.9     .05       0
Bank Sta=5005.7,5011.9
XS Rating Curve= 0 ,0
Exp/Cntr=0.3,0.1

Type RM Length L Ch R = 1 ,72587   ,582,582,582
BEGIN DESCRIPTION:
X18093
END DESCRIPTION:
XS GIS Cut Line= 3
      2502727.24     13811660.18      2502506.09     13810487.15
      2501996.49     13809516.03
#Sta/Elev= 30
  3477.2  401.42  3543.9  400.73  3946.8  397.96  4133.7  397.99  4718.5  394.18
  4788.7  392.81    4880  392.64    4902  391.45  4933.1  393.28  4978.2  392.81
  4984.6  391.66  4987.1  387.27  4987.6  386.77  4993.4  387.27    4997  388.95
  5010.4  392.85  5028.7  395.42  5050.7  395.66  5111.3  402.45  5243.6  412.38
  5271.9  415.98  5309.7  418.04  5339.7  421.56  5391.6  426.04  5452.5  430.73
  5486.4  434.81  5502.6  435.25    5541  438.69  5651.3  443.11  5767.6  445.94
#Mann= 9 ,-1 , 0
  3477.2     .07       0  3543.9     .05       0  4788.7      .1       0
  4987.1     .05       0  4993.4      .1       0    4997     .05       0
  5010.4     .07       0  5339.7     .05       0  5391.6     .07       0
Bank Sta=4987.1,4993.4
XS Rating Curve= 0 ,0
Exp/Cntr=0.3,0.1

Type RM Length L Ch R = 1 ,72005   ,469,469,469
BEGIN DESCRIPTION:
BALDRIDGE CREEK 73.0
END DESCRIPTION:
XS GIS Cut Line= 3
      2502784.92     13811448.63        2502825.       13810075.
      2502698.39     13809314.18
#Sta/Elev= 30
  3625.7  399.83  4119.5  396.29  4359.6  395.94  4419.7  394.27  4699.8  393.42
  4757.2  391.32  4779.8   390.3  4831.7  391.76  4859.9  390.64  4939.9  390.99
  4979.9  389.58  4989.9  390.53  5002.5  389.82  5006.9   385.1  5007.4   384.6
  5013.3   385.1  5020.2  387.78  5032.9  390.17  5060.7  392.12  5111.4  393.18
  5141.8  397.07  5154.6  397.49    5177  401.56  5202.7  405.44  5222.9  405.82
  5243.2  404.76  5293.9  407.19  5580.7   427.2  5709.5  433.13  5771.2  434.17
#Mann= 5 ,-1 , 0
  3625.7     .05       0  4757.2      .1       0  5006.9     .05       0
  5013.3      .1       0    5177     .07       0
Bank Sta=5006.9,5013.3
XS Rating Curve= 0 ,0
Exp/Cntr=0.3,0.1

Type RM Length L Ch R = 1 ,71536   ,470,470,470
BEGIN DESCRIPTION:
BALDRIDGE CREEK 72.0
END DESCRIPTION:
XS GIS Cut Line= 3
        2503125.       13811275.        2503225.       13810275.
        2503225.     13809874.99
#Sta/Elev= 30
  3995.1  398.97  4248.9  397.65  4650.9  392.73  4738.8  393.46  4819.2  392.22
  4889.5  390.12  4966.2   389.6    4980  389.57  4997.6  386.74  5002.6  386.74
  5010.1  388.51  5020.1  386.57  5026.8  383.09  5027.3  382.59  5033.3  383.09
  5040.1  385.96  5050.1  387.79  5060.1   387.7  5070.1  389.17  5090.1  389.19
  5100.1  387.39  5110.1  389.41  5120.1  390.31  5240.1  389.39  5250.1  390.17
  5270.1  393.28  5290.1  397.19  5310.1  399.17  5334.9  400.17  5400.1  404.81
#Mann= 5 ,-1 , 0
  3995.1     .05       0  4966.2      .1       0  5026.8     .05       0
  5033.3      .1       0  5334.9     .07       0
Bank Sta=5026.8,5033.3
XS Rating Curve= 0 ,0
Exp/Cntr=0.3,0.1

Type RM Length L Ch R = 1 ,71066   ,477,477,477
BEGIN DESCRIPTION:
BALDRIDGE CREEK 71.0
END DESCRIPTION:
XS GIS Cut Line= 3
      2503274.99     13811025.02        2503625.       13810275.
      2503474.99     13809874.98
#Sta/Elev= 30
  4172.4  397.51  4449.1  393.64  4641.7  391.95  4691.1  390.54  4735.2  388.04
  4797.5  388.31  4856.6  386.24  4861.7  386.82  4900.8  388.35  4933.9  387.66
  4940.2  386.21  4945.7   386.4  4955.9  384.89    4963  382.73  4968.5  384.73
  4985.9  382.44  4991.4  383.48  4994.1  382.42  4994.6  381.92  5000.6  382.42
  5002.7  382.42  5009.9  386.57  5015.2  384.47  5045.5  387.93  5085.5  387.01
  5149.6   390.5  5186.1  390.59  5301.8   395.9    5344  398.91  5427.3  404.32
#Mann= 6 ,-1 , 0
  4172.4     .05       0  4641.7     .07       0  4861.7      .1       0
  4994.1     .05       0  5000.6      .1       0    5344     .07       0
Bank Sta=4994.1,5000.6
XS Rating Curve= 0 ,0
Exp/Cntr=0.3,0.1

Type RM Length L Ch R = 1 ,70589   ,450,450,450
BEGIN DESCRIPTION:
BALDRIDGE CREEK 70.0
END DESCRIPTION:
XS GIS Cut Line= 3
        2504675.     13811624.99        2504025.       13810075.
        2504025.     13809824.96
#Sta/Elev= 30
  3318.4  405.91  3515.7  400.34  3568.6  397.61    3622   397.1  3654.5  395.28
  3740.5  393.48  4546.3  388.81  4600.9  388.36    4663  384.87  4671.8  385.81
  4677.6  384.73  4701.4  386.01  4706.8  383.63  4725.2  385.82  4730.6  384.61
  4814.8  385.97  4825.7  383.88  4836.5  385.53  4847.4  382.72  4854.9   385.7
  4860.3  382.69  4878.6  386.43  5001.7  386.65  5009.2  386.01  5015.4  382.48
  5015.9  381.98    5023  382.48  5039.2  385.76  5084.9  391.44  5249.2  399.49
#Mann= 6 ,-1 , 0
  3318.4     .05       0  4546.3     .07       0  4671.8      .1       0
  5015.4     .05       0    5023      .1       0  5084.9     .07       0
Bank Sta=5015.4,5023
XS Rating Curve= 0 ,0
Exp/Cntr=0.3,0.1

Type RM Length L Ch R = 1 ,70139   ,1351,1351,1351
BEGIN DESCRIPTION:
BALDRIDGE CREEK 69.0
END DESCRIPTION:
XS GIS Cut Line= 3
      2505575.02     13811125.01        2504375.       13810125.
      2504074.98     13809724.98
#Sta/Elev= 30
  3432.7   406.1    3639  401.73  3674.2  399.15  3951.5  391.34  4172.5  388.45
    4301   387.9  4351.3  387.49  4426.8  386.66  4512.5  385.49  4554.1  382.81
  4703.8  382.16  4710.3  380.77  4724.7  383.42  4746.8  383.95  4805.5  382.54
  4824.9  381.83  4831.4  384.22  4838.6  384.38  4866.6  384.55  4874.4   382.7
  4895.2     385  4961.2  385.16  4997.9  384.76  5004.5  380.54    5005  380.04
  5012.2  380.54  5031.2  384.67  5044.8  385.55  5287.5  392.56  5494.8  404.04
#Mann= 9 ,-1 , 0
  3432.7     .05       0  4172.5     .07       0    4301     .05       0
  4351.3     .07       0  4426.8     .05       0  4805.5      .1       0
  4961.2     .07       0  5004.5     .05       0  5012.2     .07       0
Bank Sta=5004.5,5012.2
XS Rating Curve= 0 ,0
Exp/Cntr=0.3,0.1

Type RM Length L Ch R = 1 ,68788   ,457,457,457
BEGIN DESCRIPTION:
BALDRIDGE CREEK 68.0
END DESCRIPTION:
XS GIS Cut Line= 3
      2505575.02     13810775.03        2505025.       13810025.
      2504275.04     13809475.03
#Sta/Elev= 30
  4074.3   400.7    4368  391.29    4682  385.41  4846.6  385.79  4893.5  383.35
  4946.9  380.87  5011.8  381.87  5026.4  380.89  5032.6  382.53    5054  382.63
  5061.9  379.37  5068.1  382.21  5076.5  378.22  5086.7  376.47  5087.2  375.97
  5095.6  376.47  5103.6  382.52  5131.5  382.62  5254.1  385.83  5276.9  385.09
  5354.4  386.56  5369.1  389.06  5376.4  392.23  5383.7  392.45  5389.9  392.21
  5398.4  388.88  5512.8  388.27  5534.2  390.77  5670.1  394.29  5934.4  404.74
#Mann= 7 ,-1 , 0
  4074.3     .05       0  4893.5      .1       0  5011.8     .07       0
  5086.7     .05       0  5095.6     .07       0  5131.5     .05       0
  5276.9     .07       0
Bank Sta=5086.7,5095.6
XS Rating Curve= 0 ,0
Exp/Cntr=0.3,0.1

Type RM Length L Ch R = 1 ,68331   ,708,708,708
BEGIN DESCRIPTION:
BALDRIDGE CREEK 67.0
END DESCRIPTION:
XS GIS Cut Line= 3
      2505675.01     13810325.01        2505275.       13809725.
        2504525.       13809425.
#Sta/Elev= 30
  4278.4  391.84  4466.2  387.84  4523.3  387.78  4602.9  385.26  4746.4  383.09
  4775.7  383.14  4817.2  381.93  4826.8  382.14  4847.8   380.9  4883.8   382.1
  4963.5  382.02    4986  381.06  4987.6  374.73  4988.1  374.23    4996  374.23
  4996.5  374.73  5002.2  375.11  5008.9  380.46  5022.1  381.36  5043.9  382.85
    5122  382.82  5391.3  386.53  5570.3  390.84  5577.1  391.66  5601.3  392.43
  5624.2   392.5  5699.6  396.22    5709  395.92    5775  398.55  5807.3  399.03
#Mann= 6 ,-1 , 0
  4278.4     .05       0  4746.4     .07       0  4817.2      .1       0
  4987.6     .05       0  4996.5      .1       0  5022.1     .05       0
Bank Sta=4987.6,4996.5
XS Rating Curve= 0 ,0
Exp/Cntr=0.3,0.1

Type RM Length L Ch R = 1 ,67623   ,428,428,428
BEGIN DESCRIPTION:
BALDRIDGE CREEK 66.0
END DESCRIPTION:
XS GIS Cut Line= 3
      2506074.99     13810024.99      2505803.93     13809554.53
        2504725.       13809175.
#Sta/Elev= 30
  4561.3  389.33  4827.6  385.49    4943  381.17  4965.2  378.03  4971.5  375.48
  4972.7  374.16  4973.2  373.66  4981.7  374.16  4987.2  378.53  4999.8  380.17
    5046   381.1  5067.7  379.31  5080.6  380.32  5118.5  380.74  5124.3  379.37
  5134.9  378.45  5205.7  380.53  5336.3  380.64  5453.8  382.47  5685.7  383.34
  5834.6  385.83  5845.8  386.77    6010  389.15  6108.9  391.65  6175.9   393.7
    6195  395.48  6201.5  393.84  6206.8   393.6  6233.2  394.94    6248  395.57
#Mann= 9 ,-1 , 0
  4561.3     .05       0  4827.6     .07       0    4943      .1       0
  4972.7     .05       0  4981.7      .1       0  5205.7     .05       0
    6010     .07       0  6108.9     .05       0  6233.2     .07       0
Bank Sta=4972.7,4981.7
XS Rating Curve= 0 ,0
Exp/Cntr=0.3,0.1

Type RM Length L Ch R = 1 ,67195   ,575,575,575
BEGIN DESCRIPTION:
BALDRIDGE CREEK 65.0
END DESCRIPTION:
XS GIS Cut Line= 3
      2506674.96     13809424.99      2505832.77     13809237.24
      2504674.96       13809125.
#Sta/Elev= 30
  4334.6  389.34  4566.2  385.06  4918.5  381.66    4939  380.86  4954.7  378.21
  4959.8  379.01  4985.4  374.34  4985.9  373.84  4995.1  374.34  4998.2  378.79
  5003.3  377.48  5010.8  379.21    5067  378.86  5095.4  379.52  5123.5  377.73
  5133.7   378.8  5201.1  378.82  5276.6  378.39  5366.3  380.01  5416.3  381.45
  5436.3  380.53  5526.8  381.18    5567  382.58  5627.2  382.39  6029.1  387.73
    6220  392.82  6250.1  395.01  6270.2  393.38  6337.9  396.03  6360.7  396.59
#Mann= 8 ,-1 , 0
  4334.6     .05       0  4566.2     .07       0  4985.4     .05       0
  4995.1     .07       0    5067      .1       0  5201.1     .07       0
  5366.3     .05       0  6337.9     .07       0
Bank Sta=4985.4,4995.1
XS Rating Curve= 0 ,0
Exp/Cntr=0.3,0.1

Type RM Length L Ch R = 1 ,66620   ,984,984,984
BEGIN DESCRIPTION:
X18092
END DESCRIPTION:
XS GIS Cut Line= 3
      2506842.28     13809006.48      2505765.47      13808814.2
      2505005.92     13809025.72
#Sta/Elev= 30
  4095.9   390.1  4377.6  384.66    4408  385.12  4499.5  383.19  4550.9  383.11
  4580.7  382.75  4591.9  381.84  4601.1  382.39  4611.2  381.62  4699.6  381.59
  4704.7  380.59  4733.1  380.11  4789.8   376.6  4834.7  377.38  4844.8  376.88
  4865.2  377.84  4885.5  377.17    4916  377.87    4984  377.57  5002.5  373.94
    5003  373.44  5012.3  373.94  5013.8  374.06    5048     379  5113.3  378.41
  5355.8  379.79  5694.8  384.29  5709.3  383.93  5792.3  386.17  5978.2  389.29
#Mann= 7 ,-1 , 0
  4095.9     .05       0  4550.9     .07       0  4789.8      .1       0
  5002.5     .05       0  5012.3      .1       0  5013.8     .07       0
  5113.3     .05       0
Bank Sta=5002.5,5012.3
XS Rating Curve= 0 ,0
Exp/Cntr=0.3,0.1

Type RM Length L Ch R = 1 ,65636   ,470,470,470
BEGIN DESCRIPTION:
BALDRIDGE CREEK 64.0
END DESCRIPTION:
XS GIS Cut Line= 3
      2506774.97       13808375.        2506325.       13808325.
      2505124.99     13808925.01
#Sta/Elev= 30
  4547.4  385.75  4733.9   382.3  4869.3  380.83  4959.9  377.53  4990.1  374.65
  5008.5  374.76  5014.1  372.69  5030.9  371.76  5053.2  373.95  5075.6  375.04
  5081.2  374.56    5098  375.42  5103.6  373.17  5111.9  375.44  5246.1  375.89
  5268.5  375.41  5276.9  373.05  5277.4  371.18  5277.9  370.68  5287.4  371.18
  5290.8  371.67  5299.2  374.64  5304.8  375.54  5327.2  377.57  5349.5  378.36
    5440  378.09  5550.8  377.97  5796.7  379.37  6087.4  382.47  6341.8  387.28
#Mann= 5 ,-1 , 0
  4547.4     .05       0  4733.9     .07       0  5277.4     .05       0
  5287.4     .07       0    5440     .05       0
Bank Sta=5277.4,5287.4
XS Rating Curve= 0 ,0
Exp/Cntr=0.3,0.1

Type RM Length L Ch R = 1 ,65166   ,443,443,443
BEGIN DESCRIPTION:
BALDRIDGE CREEK 63.0
END DESCRIPTION:
XS GIS Cut Line= 3
      2506724.99       13808125.        2506225.       13807925.
      2505024.96     13808925.03
#Sta/Elev= 30
  4466.8  384.14  4549.5  382.01    4596  382.29  4618.9  380.47  4660.7  378.98
  4667.4  379.63    4697  378.92  4726.6  377.68  4775.1  373.45  4799.3  374.46
  4811.4  373.37  4834.3  374.59  4883.5  374.54  4983.8  374.47  5008.6  373.19
  5012.5  371.41    5019  371.09  5028.2  368.66  5028.7  368.16  5038.3  368.66
  5042.2  369.23  5055.4  370.93  5061.9  370.72  5069.7  374.02  5125.7   374.8
  5197.3  377.54  5399.8  377.03    5580   377.2  6169.7   382.1  6567.4  389.66
#Mann= 7 ,-1 , 0
  4466.8     .05       0  4549.5     .07       0  4883.5     .12       0
  5028.2     .05       0  5038.3     .12       0  5042.2     .07       0
  5399.8     .05       0
Bank Sta=5028.2,5038.3
XS Rating Curve= 0 ,0
Exp/Cntr=0.3,0.1

Type RM Length L Ch R = 1 ,64723   ,429,429,429
BEGIN DESCRIPTION:
BALDRIDGE CREEK 62.0
END DESCRIPTION:
XS GIS Cut Line= 3
      2506774.96       13807675.        2506225.       13807625.
      2505024.99     13808825.01
#Sta/Elev= 30
    4443  383.46    4571  380.26  4799.6  374.98  4844.6   374.4  4854.7  373.71
  4864.7  374.03  4874.7  372.18  4884.8   371.6  4894.8   372.9  4904.9  373.06
  4914.9   371.4  4924.9  372.56  4965.1   372.4  4975.1  371.82  4985.2  369.97
  4987.7  367.58  4988.2  367.08  4997.3  367.08  4997.8  367.58  5009.4  368.66
  5023.5  368.89  5037.7  372.33  5051.8  372.63  5221.5     374  5249.8  375.44
  5513.1   376.8  6013.5  379.47  6253.9   381.6  6550.9  385.43  6692.3  388.21
#Mann= 6 ,-1 , 0
    4443     .07       0    4571     .12       0  4799.6     .07       0
  4987.7     .05       0  4997.8     .07       0  5513.1     .05       0
Bank Sta=4987.7,4997.8
XS Rating Curve= 0 ,0
Exp/Cntr=0.3,0.1

Type RM Length L Ch R = 1 ,64294   ,735,735,735
BEGIN DESCRIPTION:
BALDRIDGE CREEK 61.0
END DESCRIPTION:
XS GIS Cut Line= 3
      2506775.03     13807625.01        2505975.       13807375.
      2504774.98     13808475.02
#Sta/Elev= 30
  4166.1  384.18  4287.7  380.21  4341.7  379.03  4511.9  374.27  4550.1  375.34
    4669  370.97  4700.5  372.58  4782.7  372.17  4794.7  369.15  4805.2  371.83
  4820.4  372.53  4972.9  372.17  5001.7  368.45  5011.4  370.06    5013  367.87
  5013.5  367.37  5023.3  367.87  5025.6  373.56  5032.3  372.35  5039.7  374.85
  5074.9  376.16  5089.1  375.29  5096.5  372.95  5145.8  375.77  5180.9  374.37
  5237.7  376.45  5418.8  377.23  6214.4  381.76  6462.3  386.19  6632.2  392.68
#Mann= 6 ,-1 , 0
  4166.1     .07       0  4287.7     .12       0  4341.7     .07       0
    5013     .05       0  5023.3     .07       0  5418.8     .05       0
Bank Sta=5013,5023.3
XS Rating Curve= 0 ,0
Exp/Cntr=0.3,0.1

Type RM Length L Ch R = 1 ,63559   ,597,597,597
BEGIN DESCRIPTION:
X18091
END DESCRIPTION:
XS GIS Cut Line= 3
      2507303.82     13807295.08      2506275.05     13806977.79
      2505005.93     13807516.21
#Sta/Elev= 30
  4120.8  401.62  4391.7  393.38  4712.8  379.67  4914.1   374.6  4977.7  369.08
  4984.6  366.63  4989.8  368.37  4993.4  365.11  4993.9  364.61  5003.9  365.11
  5021.1  369.07  5040.5  370.59  5082.9     371  5125.7  371.09  5145.1  366.45
  5153.2  366.22  5158.4  370.53    5185  371.59  5219.2  373.45  5320.7  373.21
  5332.1  371.23  5355.8  371.37  5361.2  373.62  5379.5  372.93  5408.6  374.63
  5501.6  373.63  5508.7  374.69  5514.1   373.7  5754.6  375.39    6576  380.39
#Mann= 8 ,-1 , 0
  4120.8     .07       0  4993.4     .05       0  5003.9     .07       0
  5021.1     .12       0  5082.9     .07       0    5185     .12       0
  5320.7     .07       0  5754.6     .05       0
Bank Sta=4993.4,5003.9
XS Rating Curve= 0 ,0
Exp/Cntr=0.3,0.1

Type RM Length L Ch R = 1 ,62962   ,427,427,427
BEGIN DESCRIPTION:
BALDRIDGE CREEK 60.0
END DESCRIPTION:
XS GIS Cut Line= 3
      2506724.97       13806575.        2506275.       13806575.
      2505275.02     13807274.99
#Sta/Elev= 30
    4550  378.68    4700  375.63    4740  373.54  4773.5  369.73    4860  369.66
    4880  368.13    4900   369.6    4960  368.71    4980  366.84    4990  366.79
  5002.1  363.33  5002.6  362.83  5012.7  363.33  5013.5   364.5  5022.2  365.44
  5026.8  367.79  5028.3  368.56  5043.1  368.85    5058  371.44  5099.8  372.25
  5200.9  372.37  5302.1  374.27  5358.8  373.94  5366.2  374.66  5394.5  374.08
  5641.3  375.47  5708.9  375.65    5957   376.6  6040.6  377.65  6220.6  378.14
#Mann= 8 ,-1 , 0
    4550     .07       0  4773.5     .12       0  5002.1     .05       0
  5012.7     .12       0  5026.8     .07       0  5641.3     .05       0
  5708.9     .07       0    5957     .05       0
Bank Sta=5002.1,5012.7
XS Rating Curve= 0 ,0
Exp/Cntr=0.3,0.1

Type RM Length L Ch R = 1 ,62535   ,428,428,428
BEGIN DESCRIPTION:
BALDRIDGE CREEK 59.0
END DESCRIPTION:
XS GIS Cut Line= 3
      2506725.04       13806275.        2506325.       13806225.
      2505225.01     13807124.99
#Sta/Elev= 30
  4597.3  378.96  4627.7  378.33  4715.8  374.28  4720.8  374.99    4809  371.61
  4869.4  368.18  4939.3  366.99  4980.3  367.32  4990.4  366.46  4992.6  362.59
  4993.1  362.09  5003.3  362.59  5028.4  363.71  5036.3  367.79  5042.8  368.88
  5067.1  367.75  5085.9   367.3  5106.7  369.13  5114.6  367.99  5128.9  368.08
  5135.4  366.25  5149.8  367.81    5228  368.91  5266.5  371.28  5298.3  370.69
  5398.8  372.86  5707.2  374.96  6299.5  377.16  6354.2  377.47  6421.7  377.73
#Mann= 10 ,-1 , 0
  4597.3     .07       0  4627.7     .12       0  4939.3     .07       0
  4992.6     .05       0  5003.3     .07       0  5067.1     .12       0
  5266.5     .07       0  5707.2     .05       0  6299.5     .07       0
  6354.2     .05       0
Bank Sta=4992.6,5003.3
XS Rating Curve= 0 ,0
Exp/Cntr=0.3,0.1

Type RM Length L Ch R = 1 ,62107   ,539,539,539
BEGIN DESCRIPTION:
X18090
END DESCRIPTION:
XS GIS Cut Line= 3
      2507044.18     13805900.94      2506121.22     13805891.33
      2504813.62     13806785.49
#Sta/Elev= 30
  4080.6  384.38  4209.8  382.63  4325.5  379.43  4389.8  377.49  4499.8  375.67
  4529.8  374.13  4643.7  372.33    4678  372.14  4749.8  370.92  4829.8  367.18
  4979.8  367.35  5003.6  364.48  5004.3  363.33  5005.8  360.87  5006.3  360.37
  5016.5  360.87  5018.1  364.58  5024.1  366.04  5047.5  367.72  5068.9  367.43
  5122.8  368.97  5125.2  368.97  5155.6  370.71  5161.6  370.09  5191.5  370.65
    5205  371.71  5536.6  373.72  6361.3  376.57  6551.8  377.95  6587.7  378.66
#Mann= 12 ,-1 , 0
  4080.6     .07       0  4325.5     .12       0  4643.7     .07       0
    4678     .12       0  5004.3     .07       0  5005.8     .05       0
  5016.5     .07       0  5122.8     .12       0  5125.2     .07       0
  5536.6     .05       0  6361.3     .07       0  6551.8     .05       0
Bank Sta=5005.8,5016.5
XS Rating Curve= 0 ,0
Exp/Cntr=0.3,0.1

Type RM Length L Ch R = 1 ,61568   ,751,751,751
BEGIN DESCRIPTION:
BALDRIDGE CREEK 58.0
END DESCRIPTION:
XS GIS Cut Line= 3
      2506996.16     13805660.58      2505976.99      13805410.6
      2504842.48     13806304.75
#Sta/Elev= 30
  3884.8  382.94    3914  381.93  4030.1  379.84    4227  374.04  4429.8  370.93
  4534.7  370.59  4642.8   367.2  4674.9   367.8  4802.4  364.67    4823  365.21
  4843.6   363.5  4855.9  365.41  4974.9  365.69  4987.8  364.24  4990.5  360.84
    4991  360.34  5001.4  360.84  5016.7  365.06  5041.5  365.95  5095.3   369.6
  5153.1  370.33  5188.4  369.37  5209.2  371.02  5244.6  371.21  5860.8  373.94
  6092.7  374.43  6134.3  375.42  6175.8  374.55  6251.4  374.94  6378.7  375.47
#Mann= 10 ,-1 , 0
  3884.8     .12       0    3914     .05       0  4674.9     .12       0
  4990.5     .05       0  5001.4     .12       0  5041.5     .07       0
  5244.6     .05       0  5860.8     .07       0  6175.8     .05       0
  6251.4     .07       0
Bank Sta=4990.5,5001.4
XS Rating Curve= 0 ,0
Exp/Cntr=0.3,0.1

Type RM Length L Ch R = 1 ,60817   ,604,604,604
BEGIN DESCRIPTION:
BALDRIDGE CREEK 57.0
END DESCRIPTION:
XS GIS Cut Line= 3
      2506975.02     13805325.01      2506332.74     13805131.77
      2505063.61     13804785.65
#Sta/Elev= 30
  4218.2  380.36  4427.1  373.55  4500.2  374.37  4651.8  370.48  4695.2  371.43
  4704.8  371.44  4796.4  369.23    4928  367.51  4959.1  364.47    4968  360.51
  5000.6  360.62  5006.1  359.15  5006.6  358.65  5019.7  359.15  5047.5   364.7
  5073.2  363.49  5093.9  365.14  5145.7  364.73  5156.1   364.4  5161.5  361.34
  5166.7  361.08  5187.2  364.61  5205.5  364.49  5270.7  364.52  5341.4     364
  5435.9  363.05  5591.6  367.59  5798.7  371.49  5935.8  371.87  6204.4  373.68
#Mann= 11 ,-1 , 0
  4218.2     .05       0  4695.2    .063       0  4704.8     .05       0
  4796.4      .1       0  5006.1     .05       0  5019.7      .1       0
  5205.5     .12       0  5270.7      .1       0  5341.4     .12       0
  5591.6     .07       0  5935.8    .035       0
Bank Sta=5006.1,5019.7
XS Rating Curve= 0 ,0
Exp/Cntr=0.3,0.1

Type RM Length L Ch R = 1 ,60213   ,601,601,601
BEGIN DESCRIPTION:
BA21633
END DESCRIPTION:
XS GIS Cut Line= 4
      2507034.51      13804882.8      2506659.19      13804378.2
      2505712.56     13804707.65      2505088.56     13804765.89
#Sta/Elev= 30
  3590.5  377.66  3830.8  371.24  3946.4  368.25    4024  368.35  4052.8  367.15
  4101.5  367.83  4222.1  366.75    4227  367.41  4501.5  367.04  4700.3  365.97
    4785  364.63  4807.2  365.17    4833  363.65  4889.9   362.8    4965  364.15
  4996.7  362.83  5007.3     361  5012.7  358.02  5013.2  357.52  5026.4  358.02
  5028.5   359.9  5039.1  361.39  5076.4  365.01  5113.2  367.31  5354.7  368.74
  5410.1  370.93    5621  371.64  5711.4  372.86  5741.5  372.24  5848.4  373.92
#Mann= 5 ,-1 , 0
  3590.5    .035       0  3830.8     .05       0  4101.5    .035       0
  5012.7    .035       0  5026.4    .035       0
Bank Sta=5012.7,5026.4
XS Rating Curve= 0 ,0
Exp/Cntr=0.3,0.1

Type RM Length L Ch R = 1 ,59612   ,766,766,766
BEGIN DESCRIPTION:
BA13179
END DESCRIPTION:
XS GIS Cut Line= 4
      2508064.59     13803710.97      2507080.38     13803740.17
      2506062.85     13804123.82      2504665.88     13804595.04
#Sta/Elev= 30
  2834.7  374.41  3018.8  372.93  3096.3  371.67  3240.1  369.02  3384.5  371.66
    3473  366.28    3478  368.65  3574.6  363.14  3615.4   364.3  3654.6  367.17
  3724.7  364.09  4263.8  364.97  4708.9  362.65  4991.5  362.44  5010.1  360.91
  5010.6  356.71  5011.1  356.21  5024.8  356.71  5062.8  359.75  5094.5  357.92
    5105  362.93  5155.2  361.64  5377.2  364.46  5421.5  368.19  5547.6  368.88
  5661.3  370.44  5736.5  371.75  5841.5   372.2  6374.8  378.67  6381.1  378.72
#Mann= 16 ,-1 , 0
  2834.7    .094       0  3018.8    .063       0  3096.3    .094       0
  3240.1    .035       0  3615.4    .063       0  4263.8     .12       0
  4708.9    .063       0  5010.6    .063       0  5024.8    .063       0
  5155.2     .12       0  5377.2    .063       0  5547.6     .07       0
  5661.3    .035       0  5736.5     .07       0  5841.5     .05       0
  6374.8    .035       0
Bank Sta=5010.6,5024.8
XS Rating Curve= 0 ,0
Exp/Cntr=0.3,0.1

Type RM Length L Ch R = 1 ,58846   ,674,674,674
BEGIN DESCRIPTION:
X18088
END DESCRIPTION:
XS GIS Cut Line= 3
      2507717.24     13804112.61        2507025.     13803612.65
      2505179.49     13803372.35
#Sta/Elev= 30
  3339.6   375.3    3375  374.79  3805.1  366.26  3854.4  370.57  3870.1   371.6
  3889.8  368.84  3934.5  363.21  3970.7  367.24  3991.5  364.23  4191.4  363.67
  4348.7  363.48  4631.3  363.42    4970  361.61  4979.6  356.71  4980.1  356.21
    4994  356.71  5030.5     360  5141.4   358.7  5181.8  361.18    5212  359.33
    5219  362.49  5334.4  366.51  5494.4   369.5  5530.2  375.54  5585.2  373.84
  5615.4  377.52  5635.6  374.74  5736.7  376.06  5873.9  379.61  6054.6  385.75
#Mann= 13 ,-1 , 0
  3339.6    .094       0    3375    .063       0  3854.4    .035       0
  3889.8    .063       0  4191.4    .035       0  4348.7    .063       0
  4631.3     .12       0  4979.6     .05       0    4994     .12       0
  5141.4    .035       0  5334.4     .07       0  5736.7     .05       0
  5873.9     .07       0
Bank Sta=4979.6,4994
XS Rating Curve= 0 ,0
Exp/Cntr=0.3,0.1

Type RM Length L Ch R = 1 ,58172   ,588,588,588
BEGIN DESCRIPTION:
BALDRIDGE CREEK 55.0
END DESCRIPTION:
XS GIS Cut Line= 3
      2507784.55      13804045.3      2506630.79     13803074.23
      2505968.67      13802661.6
#Sta/Elev= 30
  3379.2  375.74  3478.7  373.31  3629.8  370.82  3783.8  366.74  3819.3  370.05
  3833.7  371.51  3903.9   363.1    3926  366.32  3984.3     365  4430.9  362.55
  4583.8  361.66  4628.3  357.92  4634.9  360.92  4642.6  358.56  4649.2  362.01
  4685.5     357    4735  357.36  4770.1  361.37  4855.6  358.16    4992  360.21
  5005.9  353.74  5006.4  353.24  5020.5  353.74  5043.9  356.94  5086.4  371.14
  5107.6  373.35  5286.8  379.96  5319.9  380.93  5651.1  383.79  5667.4  386.86
#Mann= 12 ,-1 , 0
  3379.2    .063       0  3478.7    .094       0  3629.8    .063       0
  3819.3    .035       0  3984.3    .063       0  4430.9    .035       0
  4583.8     .12       0  5005.9     .05       0  5020.5     .12       0
  5286.8    .035       0  5319.9     .12       0  5651.1     .07       0
Bank Sta=5005.9,5020.5
XS Rating Curve= 0 ,0
Exp/Cntr=0.3,0.1

Type RM Length L Ch R = 1 ,57584   ,423,423,423
BEGIN DESCRIPTION:
BALDRIDGE CREEK 54.0
END DESCRIPTION:
XS GIS Cut Line= 3
        2507775.     13803975.01        2506975.       13802975.
      2506475.03     13802475.03
#Sta/Elev= 30
  3719.4  375.01  3854.7   371.2  3892.3  371.67  3909.3  370.75  4010.5  368.22
  4061.2   371.5  4125.2  362.97    4154  366.54  4167.6  364.45    4215  363.94
  4357.7   364.5  4421.2  364.31  4667.7  362.45  4670.7  362.48  4730.3  361.93
  4771.9  359.46  4864.8  362.34  4943.2  362.06  4978.4  357.99  4985.5  351.64
    4986  351.14  5000.1  351.64  5014.2  357.94  5028.3  358.71  5113.2  357.37
  5306.4  364.22  5353.6  365.02  5493.6  373.26  5655.4  383.43  5707.1  385.69
#Mann= 14 ,-1 , 0
  3719.4    .063       0  3892.3    .094       0  3909.3    .063       0
  4010.5    .035       0    4215    .063       0  4357.7    .035       0
  4421.2    .063       0  4667.7    .035       0  4670.7     .12       0
  4985.5     .05       0  5000.1     .12       0  5306.4    .035       0
  5493.6     .12       0  5655.4     .07       0
Bank Sta=4985.5,5000.1
XS Rating Curve= 0 ,0
Exp/Cntr=0.3,0.1
