HEC-RAS study Copperas Creek.prj: Copperas Creek Base Level Engineering

--- Copperas Creek.g01 (geometry) --- (continued)

Type RM Length L Ch R = 1 ,87268   ,424,424,424
BEGIN DESCRIPTION:
Cooperas Creek 103.0
END DESCRIPTION:
XS GIS Cut Line= 3
      2489075.02     13844475.02        2488475.       13843875.
      2487275.01       13844075.
#Sta/Elev= 30
    4151  448.55  4264.2   443.7  4462.2  442.19  4603.6  439.31  4730.9  433.68
  4798.1  434.27  4928.9  434.76  4957.1  436.18  4971.3  434.95  4986.9  427.25
  4987.4  426.75  5005.1  427.25  5009.7  431.67  5027.4  434.47  5032.5  432.69
  5040.1  434.28  5070.5  435.28  5141.5  434.73  5171.9  432.95    5182  430.75
  5222.6  434.78  5275.8  435.19  5364.5  439.65  5473.1  442.45  5566.4  443.56
  5680.4  445.49  5780.7  448.34  6004.9  457.69  6137.9  465.58  6216.1  470.63
#Mann= 10 ,-1 , 0
    4151     .07       0  4798.1      .1       0  4986.9     .05       0
  5005.1      .1       0  5473.1     .12       0  5566.4      .1       0
  5680.4     .12       0  5780.7    .035       0  6004.9     .12       0
  6137.9    .035       0
Bank Sta=4986.9,5005.1
XS Rating Curve= 0 ,0
Exp/Cntr=0.3,0.1

Type RM Length L Ch R = 1 ,86844   ,450,450,450
BEGIN DESCRIPTION:
Cooperas Creek 102.0
END DESCRIPTION:
XS GIS Cut Line= 3
      2489425.01       13843975.        2488825.       13843675.
      2488389.92     13843092.47
#Sta/Elev= 30
  4324.8  452.73  4377.9  448.32  4422.6  446.97  4436.6  445.08    4445  445.69
  4450.6  444.53  4512.1  441.85  4526.1  442.34  4562.4  439.84  4607.1  440.29
  4615.5  439.15  4674.2  438.58  4794.4  434.32  4808.4  434.89  4906.2  432.07
  4964.9  435.11  4994.3  433.96  4998.7  433.96  5008.4  427.38  5008.9  426.88
  5026.6  427.38  5032.1  434.28  5038.4  435.17  5132.2   432.9  5182.2  433.16
  5238.5  437.46  5259.3  437.58  5357.1  443.08  5459.4  444.39  5722.7  444.02
#Mann= 5 ,-1 , 0
  4324.8     .07       0  4994.3      .1       0  5008.4     .05       0
  5026.6      .1       0  5357.1     .12       0
Bank Sta=5008.4,5026.6
XS Rating Curve= 0 ,0
Exp/Cntr=0.3,0.1

Type RM Length L Ch R = 1 ,86394   ,470,470,470
BEGIN DESCRIPTION:
Cooperas Creek 101.0
END DESCRIPTION:
XS GIS Cut Line= 3
      2489575.02     13843825.01        2488975.       13843275.
      2488474.99     13842174.97
#Sta/Elev= 30
  4190.7  458.87  4204.6  456.99  4346.7  448.02  4396.2  445.93  4488.2  441.19
  4714.5  434.96  4757.1  432.45  4763.9  433.34  4834.8  431.58  4855.8   433.3
  4905.7  432.57  4934.1  434.34  4962.4  433.88  4976.6  432.36  4981.6  427.08
  4982.1  426.58    5000  427.08  5001.3  434.02  5013.4  434.61  5283.7  430.99
  5323.2  431.41  5382.6  434.57    5457  439.64  5502.3  442.01  5542.9  441.49
  5564.9  443.36    5577  441.85  5715.4  441.76    5957  444.88    6213  457.94
#Mann= 8 ,-1 , 0
  4190.7     .07       0  4346.7     .12       0  4396.2     .07       0
  4855.8      .1       0  4981.6     .05       0    5000      .1       0
  5382.6    .035       0    5457     .12       0
Bank Sta=4981.6,5000
XS Rating Curve= 0 ,0
Exp/Cntr=0.3,0.1

Type RM Length L Ch R = 1 ,85924   ,426,426,426
BEGIN DESCRIPTION:
Cooperas Creek 100.0
END DESCRIPTION:
XS GIS Cut Line= 3
      2489925.04     13843125.01        2489325.       13842975.
      2488524.98     13842074.97
#Sta/Elev= 30
  4381.8  479.06  4410.7  476.73  4594.4  454.79  4688.5  442.58  4763.2   436.9
  4956.5  432.51    4990  430.21  4998.2  426.81  4998.7  426.31  5016.6  426.81
  5021.6  431.36  5035.8   432.9  5106.9  431.91  5134.5  433.17  5201.6  431.38
  5219.8  432.27  5227.3  431.05  5267.9  430.64  5402.9   429.6  5489.1  431.69
  5503.3  434.53  5531.7  434.39  5616.2  439.74  5722.8  441.97  5864.5  441.49
    5893  442.51    6056  453.32    6084  453.99  6097.8  455.93  6204.5  459.09
#Mann= 9 ,-1 , 0
  4381.8     .07       0  4410.7     .12       0  4594.4     .07       0
  4956.5      .1       0  4998.2     .05       0  5016.6      .1       0
  5201.6     .07       0  5267.9    .035       0  5402.9     .12       0
Bank Sta=4998.2,5016.6
XS Rating Curve= 0 ,0
Exp/Cntr=0.3,0.1

Type RM Length L Ch R = 1 ,85498   ,428,428,428
BEGIN DESCRIPTION:
Cooperas Creek 99.0
END DESCRIPTION:
XS GIS Cut Line= 3
      2490075.01     13842925.01        2489525.       13842625.
      2489275.01     13842125.02
#Sta/Elev= 30
    4367  504.76  4375.1  503.78  4380.8  499.92  4396.9  496.09  4402.6  492.02
  4412.6  489.09  4418.7  483.22  4434.9  472.29  4440.6  469.97  4456.7  473.92
  4462.4  472.42  4469.5  472.93  4492.3  463.08  4506.1  460.19  4661.3  446.62
  4866.2  432.94  4898.1  431.01  4970.7   432.8  4979.7  429.87  4981.5  426.51
    4982  426.01  4999.9  426.51  5001.9  431.06  5007.5  432.74  5134.7  430.08
  5208.7  429.94  5369.2  439.05  5427.6  443.58  5477.1  446.38  5552.5  446.56
#Mann= 8 ,-1 , 0
    4367     .12       0  4661.3     .07       0  4866.2      .1       0
  4981.5     .05       0  4999.9      .1       0  5134.7     .12       0
  5369.2     .07       0  5427.6    .035       0
Bank Sta=4981.5,4999.9
XS Rating Curve= 0 ,0
Exp/Cntr=0.3,0.1

Type RM Length L Ch R = 1 ,85070   ,355,355,355
BEGIN DESCRIPTION:
Cooperas Creek 98.0
END DESCRIPTION:
XS GIS Cut Line= 3
      2490074.99     13842874.98        2489725.       13842275.
      2489375.02     13842025.01
#Sta/Elev= 30
  4311.1  487.08    4314  487.08  4318.9  483.52  4334.2  477.51  4340.4  473.72
  4356.1  469.05    4369  462.53  4377.6  460.86  4392.1  461.01  4436.4  452.79
  4485.2   447.2  4602.5  437.62  4682.8  433.75  4704.7  434.28    4751  432.78
  4785.7  430.42  4879.7  431.59  4960.6  432.44  4967.1  426.01  4967.6  425.51
  4985.5  426.01  4992.1  426.87  4997.8  431.62  5002.8  432.13  5138.3  429.46
  5199.9  430.76  5244.4  433.44  5314.5  439.17  5349.8  443.15  5435.8  447.87
#Mann= 8 ,-1 , 0
  4311.1     .12       0  4602.5     .07       0  4879.7      .1       0
  4967.1     .05       0  4985.5      .1       0  5138.3     .05       0
  5244.4     .07       0  5314.5     .05       0
Bank Sta=4967.1,4985.5
XS Rating Curve= 0 ,0
Exp/Cntr=0.3,0.1

Type RM Length L Ch R = 1 ,84715   ,764,764,764
BEGIN DESCRIPTION:
X18530
END DESCRIPTION:
XS GIS Cut Line= 3
      2490279.07      13842807.9      2490006.59     13842044.94
        2489280.     13841627.15
#Sta/Elev= 30
  4078.4  490.68  4137.5  478.22    4177   465.5  4219.3  457.42  4230.1  452.97
    4262  447.88  4325.7  444.67  4389.4  436.59  4569.9  427.44  4597.9  429.95
  4712.6  428.97  4771.7  430.69  4788.4  429.25  4818.1  431.04  4875.5  429.87
  4983.6  431.73  4993.6  431.13  4996.5  426.07    4997  425.57    5015  426.07
  5028.8  430.92  5090.2  428.98  5167.2  430.23  5194.8     433    5294  438.12
  5372.8   444.7  5467.2  452.02  5537.5  455.02  5649.3  456.23  5726.7  456.43
#Mann= 11 ,-1 , 0
  4078.4     .12       0  4597.9     .07       0  4712.6     .12       0
  4818.1      .1       0  4996.5     .05       0    5015      .1       0
  5090.2     .12       0  5194.8     .07       0  5372.8     .05       0
  5537.5    .035       0  5649.3     .05       0
Bank Sta=4996.5,5015
XS Rating Curve= 0 ,0
Exp/Cntr=0.3,0.1

Type RM Length L Ch R = 1 ,83951   ,596,596,596
BEGIN DESCRIPTION:
Cooperas Creek 97.0
END DESCRIPTION:
XS GIS Cut Line= 3
      2490630.26     13842674.67      2490157.96     13841917.78
      2489382.91     13841506.03
#Sta/Elev= 30
  4488.2  460.08  4558.4  458.36  4637.5  453.08  4643.4  454.36  4688.2  451.76
  4826.2  439.71  4978.4  430.13  4990.4  424.12  4990.9  423.62  5008.9  424.12
    5015  424.66  5020.9   428.3  5042.1  429.76  5057.4  428.76  5100.7  430.24
  5180.1  430.17  5302.2  430.31    5380  430.36  5413.7   430.8  5459.1  429.77
  5523.6  430.55  5601.2   429.1    5627  429.69  5771.8   436.2  5836.7  440.44
  5849.1  439.98  5938.8  444.78  6057.6  451.28    6183  454.71    6258  454.66
#Mann= 13 ,-1 , 0
  4488.2     .12       0  4990.4     .05       0  5008.9     .12       0
  5180.1      .1       0  5302.2     .12       0    5380     .07       0
  5413.7     .12       0  5523.6      .1       0  5601.2     .07       0
    5627     .05       0  5771.8     .12       0  5938.8     .05       0
    6183    .035       0
Bank Sta=4990.4,5008.9
XS Rating Curve= 0 ,0
Exp/Cntr=0.3,0.1

Type RM Length L Ch R = 1 ,83355   ,698,698,698
BEGIN DESCRIPTION:
X18529
END DESCRIPTION:
XS GIS Cut Line= 4
      2491029.87     13842801.79      2490660.52     13841802.74
      2490036.86     13841409.16      2489329.22     13841439.41
#Sta/Elev= 30
  3715.5  471.24  3754.7  465.15    3840  457.07  3925.3  451.35  4059.9  444.34
    4217   439.1  4373.1  435.41    4533  437.88  4614.8  436.72    4641  436.75
    4747  438.06  4847.1  438.46  4937.6  435.85  4964.5  434.03  4971.8  429.25
  4987.1  427.18  4990.8  423.63  4991.3  423.13  5009.3  423.63  5023.6  428.46
  5044.8  427.25  5081.2  429.53  5123.6  428.02  5258.6  428.92    5473  428.93
  5720.2  433.62  5950.4  445.08  6103.3   450.3  6202.1  452.61  6226.4  452.92
#Mann= 11 ,-1 , 0
  3715.5     .12       0    4217     .05       0  4614.8     .07       0
    4641      .1       0    4747     .07       0  4937.6      .1       0
  4990.8     .05       0  5009.3      .1       0  5258.6     .05       0
  6103.3    .035       0  6202.1     .05       0
Bank Sta=4990.8,5009.3
XS Rating Curve= 0 ,0
Exp/Cntr=0.3,0.1

Type RM Length L Ch R = 1 ,82657   ,565,565,565
BEGIN DESCRIPTION:
Cooperas Creek 96.0
END DESCRIPTION:
XS GIS Cut Line= 3
      2491060.16      13842832.1      2490593.92     13841342.56
      2490606.03     13840355.63
#Sta/Elev= 30
  3271.1  480.49  3304.9  477.51  3310.2  474.87  3351.9  468.38  3369.8  467.87
  3375.1  465.56  3402.3  464.76  3414.8  461.19    3440  458.14  3613.8  446.47
  3794.3  438.62  4001.5  433.65  4314.4  435.75  4418.4  438.42  4522.4  437.17
  4699.7  429.37  4730.5  428.72  4959.5  427.43  4969.5  427.11  4978.8  422.15
  4979.3  421.65  5000.1  422.15  5009.5  428.44  5029.5  430.78  5227.8  428.55
  5330.4  432.77  5549.5  447.62  5729.5  455.27  5769.5  458.88  5818.9  458.83
#Mann= 11 ,-1 , 0
  3271.1     .12       0  3794.3     .05       0  4314.4     .07       0
  4418.4     .12       0  4522.4     .07       0  4699.7     .12       0
  4730.5      .1       0  4978.8     .05       0  5000.1      .1       0
  5227.8     .07       0  5330.4     .12       0
Bank Sta=4978.8,5000.1
XS Rating Curve= 0 ,0
Exp/Cntr=0.3,0.1

Type RM Length L Ch R = 1 ,82092   ,950,950,950
BEGIN DESCRIPTION:
Cooperas Creek 95.0
END DESCRIPTION:
XS GIS Cut Line= 3
      2491114.65     13842795.78        2491025.       13841525.
      2491124.99     13841125.05
#Sta/Elev= 30
  3721.9  488.83  3787.9     483    3853   473.5  3929.1  459.58  3988.3  454.13
  4123.7  443.26    4274  435.55  4304.1  438.94  4334.2  439.58  4414.4   431.2
  4434.4  431.58  4474.5  436.11    4494  430.43    4499  434.07  4504.6  430.58
  4524.7  429.12  4786.5  426.22  4975.8  427.87  4993.3  426.17  4995.5   422.8
    4996   422.3  5016.8   422.8  5026.8  426.52  5061.5  426.51  5088.6  425.31
  5137.6  428.07  5173.1  427.61  5316.1  440.37    5332  441.65  5408.1  449.57
#Mann= 8 ,-1 , 0
  3721.9     .12       0  3988.3     .05       0  4995.5     .05       0
  5016.8     .05       0  5061.5      .1       0  5173.1     .07       0
  5316.1      .1       0    5332     .07       0
Bank Sta=4995.5,5016.8
XS Rating Curve= 0 ,0
Exp/Cntr=0.3,0.1

Type RM Length L Ch R = 1 ,81142   ,686,686,686
BEGIN DESCRIPTION:
Cooperas Creek 94.0
END DESCRIPTION:
XS GIS Cut Line= 3
      2492186.39     13842517.23      2491708.03     13842014.66
        2491175.     13841174.99
#Sta/Elev= 30
  4290.7  461.75  4300.3  460.57  4328.6  462.26  4498.5  459.54  4703.6  450.88
  4780.1  445.28  4854.8  438.74  4919.7  435.34    4958  432.26  4972.2  426.39
  4972.4   420.1  4972.9   419.6  4993.9   420.1    4996  422.06  5031.2  426.32
    5067  426.06  5073.6  424.34  5079.5  425.67    5110  424.86  5173.6   427.9
  5232.9  426.74  5355.6  427.83  5407.3  426.14  5443.7  426.39  5464.9   428.4
  5507.3   427.2  5756.1  436.63  5892.7  446.05  5929.1  445.67  5979.1  448.42
#Mann= 8 ,-1 , 0
  4290.7     .12       0  4780.1     .07       0  4854.8     .05       0
  4919.7     .07       0  4972.4     .05       0  4993.9     .07       0
    4996      .1       0  5756.1     .07       0
Bank Sta=4972.4,4993.9
XS Rating Curve= 0 ,0
Exp/Cntr=0.3,0.1

Type RM Length L Ch R = 1 ,80456   ,602,602,602
BEGIN DESCRIPTION:
Cooperas Creek 93.0
END DESCRIPTION:
XS GIS Cut Line= 3
      2492025.04     13841525.01        2491575.       13841375.
      2491174.99     13841124.99
#Sta/Elev= 30
    4531  464.65  4538.8   464.3  4573.2  463.85  4594.3  461.08    4647  447.57
  4720.8  437.95  4805.1  431.67  4826.2  428.92  4865.8  427.14  4952.7  422.12
  4963.2  423.03    4984  421.01  4984.5  420.51  5005.6  421.01  5013.1  425.42
  5018.9   424.4  5028.4  426.15  5064.3  424.99  5128.6  426.05  5143.9  428.11
  5186.4   430.8    5223  430.62  5312.3  439.45  5338.5  440.65  5353.9  442.97
  5369.2  443.81  5390.4  444.59  5396.3  443.74  5418.1  446.86  5477.1   449.1
#Mann= 6 ,-1 , 0
    4531     .07       0  4538.8     .12       0  4865.8      .1       0
    4984     .05       0  5005.6      .1       0  5312.3     .07       0
Bank Sta=4984,5005.6
XS Rating Curve= 0 ,0
Exp/Cntr=0.3,0.1

Type RM Length L Ch R = 1 ,79854   ,570,570,570
BEGIN DESCRIPTION:
Cooperas Creek 92.0
END DESCRIPTION:
XS GIS Cut Line= 3
      2492074.97     13841374.97        2491575.       13840775.
        2491225.       13840975.
#Sta/Elev= 30
    4219  462.68  4261.3  459.97  4283.4  455.05  4289.9  451.86  4339.4  444.32
  4396.6  439.51  4471.9  436.15  4603.1   431.6    4691  428.41  4715.6  426.23
  4723.4  427.06  4822.3  423.22  4857.4  425.23  4921.9  425.76  4935.5  423.98
    4972   422.8  4975.5  420.31    4976  419.81  4997.1  420.31  5002.9  420.55
  5007.9  423.25    5023  424.91  5072.7     425  5110.1  429.82  5147.6  432.98
  5153.3  432.39  5169.1  435.01  5190.7  436.52  5387.3  445.45  5403.1  446.03
#Mann= 7 ,-1 , 0
    4219     .12       0  4471.9      .1       0  4603.1     .12       0
    4691      .1       0  4975.5     .05       0  4997.1      .1       0
  5387.3     .07       0
Bank Sta=4975.5,4997.1
XS Rating Curve= 0 ,0
Exp/Cntr=0.3,0.1

Type RM Length L Ch R = 1 ,79284   ,570,570,570
BEGIN DESCRIPTION:
Cooperas Creek 91.0
END DESCRIPTION:
XS GIS Cut Line= 3
      2492374.99     13840874.99        2491775.       13840275.
      2491225.02     13839925.02
#Sta/Elev= 30
    4147  459.34  4175.3  459.53  4260.1  454.81  4359.1  444.94  4500.5  436.26
  4656.1  432.63  4726.8  429.91  4824.7  421.94  4843.3  421.55  4843.8  421.05
  4864.9  421.55  4882.4  422.83  4896.5  422.57  4910.7  424.14  4967.2  425.31
  4981.4  425.39    4992  423.37  5009.1  421.99  5031.1  424.04  5054.8  424.35
  5112.3  423.11  5227.5  427.17  5252.9  429.18  5300.3  432.16  5336.7   432.9
  5409.5  436.71  5436.6  439.29  5457.8  439.33  5611.9  448.82  5647.4  449.64
#Mann= 5 ,-1 , 0
    4147     .12       0  4824.7      .1       0  4843.3     .05       0
  4864.9      .1       0  5252.9     .12       0
Bank Sta=4843.3,4864.9
XS Rating Curve= 0 ,0
Exp/Cntr=0.3,0.1

Type RM Length L Ch R = 1 ,78714   ,565,565,565
BEGIN DESCRIPTION:
Cooperas Creek 90.0
END DESCRIPTION:
XS GIS Cut Line= 3
        2492375.     13840724.99        2492175.       13840375.
        2492175.     13839575.01
#Sta/Elev= 30
  4592.9  454.43  4673.5  450.84    4703  450.77  4708.8  449.44  4740.5  447.39
  4777.2  446.93  4805.2  442.07  4811.7   439.4  4821.1  437.22  4842.7   434.2
    4870   428.5  4892.3  426.12  4938.4   425.1  4949.8  421.79  4950.3  421.29
  4971.7  421.79  4993.1  422.98  5043.7  423.39    5116  422.84    5126  423.94
    5156  424.15    5226  422.26  5266.9  425.66    5306  429.43  5358.7  431.34
    5496  439.84    5576  442.75    5626  442.86  5749.1     448    5796  450.12
#Mann= 7 ,-1 , 0
  4592.9     .12       0  4949.8     .05       0  4971.7     .12       0
  5043.7      .1       0  5266.9     .05       0  5358.7     .12       0
  5749.1     .05       0
Bank Sta=4949.8,4971.7
XS Rating Curve= 0 ,0
Exp/Cntr=0.3,0.1

Type RM Length L Ch R = 1 ,78149   ,544,544,544
BEGIN DESCRIPTION:
Cooperas Creek 89.0
END DESCRIPTION:
XS GIS Cut Line= 3
        2492475.     13840825.01        2492675.       13840175.
      2492175.01     13839475.01
#Sta/Elev= 30
    4321  456.67  4446.6  448.06  4473.4  447.93  4530.3  444.39  4551.2  441.81
    4593  439.38  4642.1   432.5    4680  431.99  4745.4  426.28  4750.6  427.33
  4778.1  424.17  4783.3  424.94  4833.7  421.99    4852  422.16  4881.4  420.97
  4886.6  422.16  4919.3  422.23  4973.8  419.09  4974.3  418.59  4995.7  419.09
  4998.5  420.35  5023.2  422.04  5087.1  420.18  5144.9  420.19  5170.8  421.85
  5316.9  430.76  5625.4  441.48  5788.8  450.48  5824.4  453.66  5861.3  454.29
#Mann= 5 ,-1 , 0
    4321     .12       0    4852      .1       0  4973.8     .05       0
  4995.7      .1       0  5170.8     .05       0
Bank Sta=4973.8,4995.7
XS Rating Curve= 0 ,0
Exp/Cntr=0.3,0.1

Type RM Length L Ch R = 1 ,77605   ,563,563,563
BEGIN DESCRIPTION:
Cooperas Creek 88.0
END DESCRIPTION:
XS GIS Cut Line= 3
      2494175.04     13840225.01        2493075.       13839875.
      2492275.01     13839475.01
#Sta/Elev= 30
  3846.7  444.56  3895.1     443  4009.8   433.9  4112.2   428.2  4214.7  422.08
  4260.1  420.74  4266.5  418.69  4292.4  421.31    4340  419.84  4381.9  420.53
    4491  419.12  4513.8  420.01  4560.7  421.31  4581.3     419  4592.9  420.78
  4657.3  419.69  4754.1  418.19  4931.9   420.8  4969.6  420.36  4979.6  417.78
  4980.1  417.28  5001.5  417.78  5023.4  420.77  5083.9  420.51  5143.6  419.86
  5216.3  421.71  5501.4  434.08  5716.6  438.95  5842.4  444.95  5895.5  449.86
#Mann= 10 ,-1 , 0
  3846.7     .07       0  4009.8    .035       0  4112.2     .07       0
  4214.7      .1       0  4513.8     .12       0  4657.3     .07       0
  4931.9      .1       0  4979.6     .05       0  5001.5      .1       0
  5083.9     .05       0
Bank Sta=4979.6,5001.5
XS Rating Curve= 0 ,0
Exp/Cntr=0.3,0.1

Type RM Length L Ch R = 1 ,77042   ,498,498,498
BEGIN DESCRIPTION:
Cooperas Creek 87.0
END DESCRIPTION:
XS GIS Cut Line= 3
        2494225.       13840075.        2493425.       13839475.
      2491974.98     13838324.99
#Sta/Elev= 30
  4004.2  456.26  4151.4  443.45  4221.5  433.33  4343.8  423.13  4404.2  420.52
  4493.2  419.27  4613.8  418.64  4734.4  417.93  4826.1   416.3  4914.5  418.59
  4926.1  418.56  4929.7  415.49  4930.2  414.99  4951.7  415.49  4954.2  417.82
  4961.5  418.53  5007.4  417.78  5017.8  419.01  5046.2  417.51  5081.9  421.44
  5160.4  423.16  5438.2  420.88  5872.1   422.7    6093  430.59  6316.3  446.83
  6442.3   456.6  6663.4  480.25  6762.8  502.53    6798  507.87  6854.9  511.46
#Mann= 12 ,-1 , 0
  4004.2     .05       0  4151.4    .035       0  4221.5     .05       0
  4343.8     .07       0  4493.2     .12       0  4613.8      .1       0
  4734.4     .07       0  4914.5      .1       0  4929.7     .05       0
  4951.7      .1       0  5046.2     .05       0  6316.3     .12       0
Bank Sta=4929.7,4951.7
XS Rating Curve= 0 ,0
Exp/Cntr=0.3,0.1

Type RM Length L Ch R = 1 ,76544   ,554,554,554
BEGIN DESCRIPTION:
Cooperas Creek 86.0
END DESCRIPTION:
XS GIS Cut Line= 3
      2494224.98     13840024.98        2493625.       13839225.
      2492625.03     13838075.04
#Sta/Elev= 30
    3984  456.96    4034  454.04    4234  430.92  4356.2  422.51  4519.4   417.9
  4623.4  418.25  4686.3  417.13  4781.6  418.42    4812  417.27  4937.6   417.4
  4939.8  417.36  5015.4  417.14  5091.6  415.66  5092.1  415.16  5116.6  415.66
  5118.3  418.04  5132.6   419.1  5210.4  421.65  5621.6  419.17  5784.9  420.62
  5841.9  423.68  5862.7  421.79  5983.3  428.83  5998.2  431.38  6089.7  437.44
    6196  448.61  6259.6  457.31  6345.1  474.78  6394.5  481.27  6507.9   488.7
#Mann= 13 ,-1 , 0
    3984     .05       0  4356.2     .07       0  4519.4    .035       0
  4623.4      .1       0  4686.3    .035       0  4781.6     .07       0
    4812      .1       0  4937.6     .12       0  4939.8      .1       0
  5015.4     .05       0  5091.6     .05       0  5116.6     .05       0
  5998.2     .12       0
Bank Sta=5091.6,5116.6
XS Rating Curve= 0 ,0
Exp/Cntr=0.3,0.1

Type RM Length L Ch R = 1 ,75990   ,563,563,563
BEGIN DESCRIPTION:
Cooperas Creek 85.0
END DESCRIPTION:
XS GIS Cut Line= 3
      2494220.85     13839943.86        2494075.       13839025.
      2493275.02     13838225.02
#Sta/Elev= 30
    4070   450.1  4074.7  448.66  4079.7  449.08  4129.6  442.15  4220.7  435.02
  4446.9  423.08  4520.7  420.28  4666.2  417.33  4847.2  416.55    4889  416.44
  4929.5  413.22  4947.2  413.63  4980.1  414.73  5016.1  413.04  5016.6  412.54
  5041.1  413.04  5056.9  415.29  5071.1  415.86  5085.2  414.13  5099.4  415.92
  5159.7  415.44  5198.3   414.6  5226.6  415.83  5573.6  416.74  5709.1   418.1
  5848.9  422.56  5919.6  426.83  6006.8  433.83  6046.9  438.47  6131.7   445.6
#Mann= 10 ,-1 , 0
    4070     .05       0  4446.9     .07       0  4847.2     .12       0
  4947.2      .1       0  5016.1     .05       0  5041.1      .1       0
  5159.7     .05       0  5573.6    .035       0  5709.1     .05       0
  6006.8     .07       0
Bank Sta=5016.1,5041.1
XS Rating Curve= 0 ,0
Exp/Cntr=0.3,0.1

Type RM Length L Ch R = 1 ,75427   ,584,584,584
BEGIN DESCRIPTION:
Cooperas Creek 84.0
END DESCRIPTION:
XS GIS Cut Line= 3
      2494875.02     13838875.01        2494275.       13838725.
      2493474.99     13838124.99
#Sta/Elev= 30
  4386.9  450.43    4418  448.88  4619.7  434.32  4648.5   432.9  4698.7  429.86
  4809.5  425.82  4904.9  420.01    4941  414.81  4946.1  415.75  4953.9   414.1
  4964.2  413.82  4969.2  410.45  4969.7  409.95  4995.2  410.45  5002.8  412.31
  5027.3  414.95  5148.1  413.62  5291.8  415.35  5527.3  415.06  5629.4  417.27
  5683.5  418.28  5748.8  421.33  5791.8  422.94  5818.9   426.7  5877.3   431.2
  5941.8  438.28  5967.6   443.1  5983.5  445.12  5991.8  448.33  6005.4  451.26
#Mann= 9 ,-1 , 0
  4386.9     .07       0    4418     .12       0  4619.7     .07       0
  4648.5     .05       0  4969.2     .05       0  4995.2     .05       0
  5629.4    .035       0  5748.8     .05       0  5967.6     .12       0
Bank Sta=4969.2,4995.2
XS Rating Curve= 0 ,0
Exp/Cntr=0.3,0.1

Type RM Length L Ch R = 1 ,74843   ,566,566,566
BEGIN DESCRIPTION:
Cooperas Creek 83.0
END DESCRIPTION:
XS GIS Cut Line= 3
      2494874.95     13838274.99        2494175.       13838175.
        2493425.       13838075.
#Sta/Elev= 30
  4292.9  458.15  4343.4  454.26    4404   445.6  4444.4   438.2  4480.9  433.86
  4535.3  427.54  4666.6   418.2  4737.3  415.12  4801.9  414.19  4828.2   413.6
  4898.9  414.46  4929.2  412.83  4949.5  413.01  4959.6  411.98  4966.7   408.1
  4967.2   407.6  4992.9   408.1  5020.1  411.71  5052.1  414.68  5070.6  413.74
  5198.2  413.92  5297.2  415.98  5393.4  421.25  5423.7  424.73  5443.9  425.14
  5514.5  430.73  5524.6  430.83  5614.8  439.33  5726.3  453.81  5756.6  455.95
#Mann= 9 ,-1 , 0
  4292.9     .12       0  4480.9     .07       0  4801.9      .1       0
  4966.7     .05       0  4992.9      .1       0  5052.1     .05       0
  5198.2    .035       0  5297.2     .05       0  5614.8     .12       0
Bank Sta=4966.7,4992.9
XS Rating Curve= 0 ,0
Exp/Cntr=0.3,0.1

Type RM Length L Ch R = 1 ,74277   ,560,560,560
BEGIN DESCRIPTION:
Cooperas Creek 82.0
END DESCRIPTION:
XS GIS Cut Line= 3
        2494925.       13838225.        2494125.       13837625.
      2493675.04     13837824.98
#Sta/Elev= 30
  4000.1   456.7  4107.4  451.07    4172  441.69  4192.8  436.92  4240.1   431.2
  4286.6  426.45  4379.9  420.33  4424.3  417.89  4522.5  414.22  4600.1  411.92
  4829.4  413.35  4907.4  414.45  4943.7   413.5    4972  409.36  4978.2  410.17
  4983.9  406.56  4984.4  406.06  5010.1  406.56    5022  412.63  5043.9  413.65
  5089.7  413.44  5107.5  411.48    5146  411.74  5211.4   413.3  5255.2  416.25
  5286.7  417.47  5333.2  422.37  5379.7  429.21  5408.4  429.99  5492.5  438.23
#Mann= 11 ,-1 , 0
  4000.1     .12       0  4240.1     .07       0  4379.9     .05       0
  4424.3     .07       0  4522.5     .05       0  4829.4      .1       0
  4943.7     .05       0  4983.9     .05       0  5010.1     .05       0
    5146    .035       0  5255.2     .12       0
Bank Sta=4983.9,5010.1
XS Rating Curve= 0 ,0
Exp/Cntr=0.3,0.1

Type RM Length L Ch R = 1 ,73717   ,560,560,560
BEGIN DESCRIPTION:
Cooperas Creek 81.0
END DESCRIPTION:
XS GIS Cut Line= 3
      2494824.99       13837175.        2494025.       13837125.
      2493624.97     13836624.97
#Sta/Elev= 30
  4198.9  434.96  4329.1  423.28  4459.4  414.97  4528.5  412.02  4602.2  409.97
    4780  412.71  4810.1  411.84  4919.4   412.4  4950.3  412.11  4960.4  412.95
  4980.4  412.17  4990.4  409.79  4997.9  406.43  5007.7  406.42  5008.9  405.59
  5009.4  405.09  5035.3  405.59  5036.5  406.88  5042.9  409.22  5064.5  412.43
  5121.3  414.25  5151.7  413.65  5179.8  415.28  5263.2  419.44  5484.7  435.37
  5491.1  437.17  5519.9  439.07  5575.5  446.35  5636.7  453.22  5640.8  453.29
#Mann= 10 ,-1 , 0
  4198.9     .07       0  4528.5     .05       0  4919.4      .1       0
  5008.9     .05       0  5035.3      .1       0  5151.7      .1       0
  5179.8     .12       0  5263.2     .07       0  5575.5     .05       0
  5636.7     .07       0
Bank Sta=5008.9,5035.3
XS Rating Curve= 0 ,0
Exp/Cntr=0.3,0.1

Type RM Length L Ch R = 1 ,73157   ,560,560,560
BEGIN DESCRIPTION:
Cooperas Creek 80.0
END DESCRIPTION:
XS GIS Cut Line= 3
      2495025.03     13837225.02        2494225.       13836675.
      2493625.04     13836575.01
#Sta/Elev= 30
  4033.9  448.45  4195.5  439.35    4307  432.38  4328.2  432.87  4393.9  425.85
  4501.4  417.52  4638.8  412.51  4744.6  410.81  4781.5  410.45  4889.8  410.24
  4895.8  411.44  4904.6   409.1  4910.7  410.21  4919.5   406.2  4963.2  405.62
  4963.7  405.12  4989.6  405.62  4991.2  407.35  5001.7  409.95  5018.3  411.35
  5111.9  411.05    5167   411.2  5211.3  413.43  5360.6  421.51  5488.1  433.05
  5519.3  440.13  5524.3  439.98  5562.4  449.95    5609  454.22    5613  454.38
#Mann= 12 ,-1 , 0
  4033.9     .05       0  4195.5     .07       0  4744.6     .05       0
  4781.5     .07       0  4963.2     .05       0  4989.6     .07       0
  5018.3     .05       0  5111.9    .035       0  5211.3     .05       0
  5360.6     .07       0  5488.1     .05       0    5609     .07       0
Bank Sta=4963.2,4989.6
XS Rating Curve= 0 ,0
Exp/Cntr=0.3,0.1

Type RM Length L Ch R = 1 ,72597   ,423,423,423
BEGIN DESCRIPTION:
Cooperas Creek 79.0
END DESCRIPTION:
XS GIS Cut Line= 3
      2494925.02       13836325.        2494525.       13836375.
      2493725.04       13836375.
#Sta/Elev= 30
  4589.3  431.64  4690.1   433.5  4712.8  433.31  4796.9  430.38  4821.1  429.34
  4861.4   425.5  4901.7  422.94  4949.6  417.19  4954.6  417.54  4982.4  412.44
  4989.9  410.27  4994.9  410.27  4999.2  403.63  4999.7  403.13  5025.2  403.13
  5025.7  403.63  5032.4   410.1  5094.6  409.65  5202.4  411.32  5291.6  409.13
  5352.4  409.84  5362.4  410.52  5390.1  410.89  5442.4  409.92  5488.7  410.92
  5552.4   412.9  5677.5  420.73  5732.4  426.95  5789.9   437.8  5792.4   437.8
#Mann= 9 ,-1 , 0
  4589.3     .05       0  4796.9     .07       0  4999.2     .05       0
  5025.7     .07       0  5094.6     .05       0  5291.6     .07       0
  5390.1    .035       0  5488.7     .05       0  5677.5     .07       0
Bank Sta=4999.2,5025.7
XS Rating Curve= 0 ,0
Exp/Cntr=0.3,0.1

Type RM Length L Ch R = 1 ,72174   ,587,587,587
BEGIN DESCRIPTION:
X18528
END DESCRIPTION:
XS GIS Cut Line= 3
      2494856.61     13836129.22      2494420.66     13836002.07
      2493494.29     13836026.29
#Sta/Elev= 30
  4500.4   430.9  4534.2  430.51    4636  426.84  4737.8  422.58    4817   419.5
  4839.6  418.61  4891.6   417.8  4954.5  413.61  4960.2  411.54  4970.2     410
  4986.9  403.49  4987.4  402.99  5012.9  402.99  5013.4  403.49  5020.2  409.34
  5030.2  409.58  5055.4  408.52  5100.2  408.72    5139  410.27  5240.3  410.15
  5270.3  408.76  5336.2  410.12  5390.3  409.21  5434.9  409.72  5490.4  410.42
  5590.4  415.53    5757  429.22  5770.5  429.31  5840.5  433.91  5881.2   438.9
#Mann= 13 ,-1 , 0
  4500.4     .05       0  4534.2    .035       0    4636     .05       0
  4737.8     .07       0    4817     .05       0  4839.6     .12       0
  4986.9     .05       0  5013.4     .12       0  5055.4     .05       0
    5139     .07       0  5336.2    .035       0  5434.9     .05       0
    5757     .07       0
Bank Sta=4986.9,5013.4
XS Rating Curve= 0 ,0
Exp/Cntr=0.3,0.1

Type RM Length L Ch R = 1 ,71587   ,720,720,720
BEGIN DESCRIPTION:
X18527
END DESCRIPTION:
XS GIS Cut Line= 4
      2494808.18     13835989.96      2494553.87     13835705.38
      2494045.26     13835584.28      2493354.97     13835687.21
#Sta/Elev= 30
  4041.8  427.73  4182.5  423.71  4323.8  421.73    4409  418.55  4504.5  411.84
  4537.9  411.25  4638.5  409.44  4709.3     409  4739.1  408.85  4831.8  409.41
    4854  408.12  4948.9  408.95  4956.7   408.4  4966.8  405.99  4970.3  403.52
  4970.8  403.02  4996.8  403.52  4997.1   407.4  5007.2  408.17  5027.4  407.17
  5067.9  409.64  5100.8  409.72  5158.9  410.53  5238.7  414.04  5255.6  415.87
  5324.9  419.19  5467.5   431.7  5514.1  435.58  5573.4   440.3  5644.2  443.74
#Mann= 11 ,-1 , 0
  4041.8     .05       0  4537.9    .035       0  4638.5     .07       0
  4709.3    .035       0  4739.1     .07       0  4970.3     .05       0
  4996.8     .07       0  5100.8    .035       0  5238.7     .05       0
  5467.5     .07       0  5514.1     .05       0
Bank Sta=4970.3,4996.8
XS Rating Curve= 0 ,0
Exp/Cntr=0.3,0.1

Type RM Length L Ch R = 1 ,70867   ,549,549,549
BEGIN DESCRIPTION:
Cooperas Creek 78.0
END DESCRIPTION:
XS GIS Cut Line= 3
      2494775.01     13835925.02        2494325.       13835175.
      2494074.98     13834774.97
#Sta/Elev= 30
  4133.4  425.64  4236.4  423.09  4358.9   421.7    4425  419.83  4455.8  417.83
  4580.5  411.43  4634.9  409.75  4689.2  409.55  4763.4  408.89  4809.8  409.07
  4899.2  406.48  4939.2  406.56  4949.8  406.06  4957.5  402.39  4963.4  403.83
  4971.2  400.02  4971.7  399.52  4998.2  400.02  5005.1  407.49  5106.4  408.44
  5161.4  410.25  5189.1  412.95  5204.4  412.62  5247.1  416.58  5298.7  420.53
  5335.3  424.73  5385.4  433.97    5399  439.85  5420.8  445.47  5479.8  451.52
#Mann= 10 ,-1 , 0
  4133.4     .05       0  4455.8     .07       0  4580.5     .05       0
  4689.2      .1       0  4763.4     .07       0  4939.2      .1       0
  4971.2     .05       0  4998.2      .1       0  5106.4     .07       0
  5247.1     .05       0
Bank Sta=4971.2,4998.2
XS Rating Curve= 0 ,0
Exp/Cntr=0.3,0.1

Type RM Length L Ch R = 1 ,70318   ,317,317,317
BEGIN DESCRIPTION:
Cooperas Creek 77.0
END DESCRIPTION:
XS GIS Cut Line= 3
        2494875.     13836024.99        2494675.       13834925.
      2494074.98     13834724.99
#Sta/Elev= 30
  3891.4  430.04  4379.3  416.99  4418.6  416.83  4623.2  412.05  4744.3  410.63
  4817.6  407.72  4917.9  407.99  4968.8  404.91  4982.7   402.2  4985.8  399.94
  4986.3  399.44  5012.8  399.94    5020  405.28  5062.1  407.26  5083.2  407.36
  5104.3  406.22  5114.8  407.28  5146.5  407.01  5246.1  408.98  5272.9  408.92
    5294  410.53  5336.2  410.55  5367.8  411.68  5404.7   414.2  5456.8  420.86
  5494.3  426.01  5515.4  430.24  5568.1  445.73  5599.7  450.29  5641.9  453.78
#Mann= 6 ,-1 , 0
  3891.4     .05       0  4744.3      .1       0  4985.8     .05       0
  5012.8      .1       0  5246.1     .07       0  5456.8     .05       0
Bank Sta=4985.8,5012.8
XS Rating Curve= 0 ,0
Exp/Cntr=0.3,0.1

Type RM Length L Ch R = 1 ,70001   ,615,615,615
BEGIN DESCRIPTION:
X18526
END DESCRIPTION:
XS GIS Cut Line= 3
       2495074.6     13835880.98       2495074.6     13835027.22
      2494414.62     13833901.01
#Sta/Elev= 30
  3852.6  426.84  4078.6  424.65  4468.6  410.79  4678.6  408.53  4824.8   409.7
  4888.5   405.2  4949.7   407.9  4969.7  406.37  4976.9  403.72  4979.1  400.37
  4979.6  399.87  5006.1  400.37  5014.1  405.02  5021.9  405.56  5029.8  404.11
  5035.6  405.66  5088.4   404.8  5234.1  408.44  5306.4  411.85  5350.1  413.59
  5446.1  418.92  5467.6  418.29  5520.3  423.75  5563.4  426.39  5569.2  425.49
  5707.9  437.29  5745.1  438.53  5862.4  450.06  5929.9  452.88  6011.7  454.61
#Mann= 8 ,-1 , 0
  3852.6     .05       0  4888.5      .1       0  4979.1     .05       0
  5006.1      .1       0  5234.1     .12       0  5306.4      .1       0
  5350.1     .12       0  5929.9    .035       0
Bank Sta=4979.1,5006.1
XS Rating Curve= 0 ,0
Exp/Cntr=0.3,0.1

Type RM Length L Ch R = 1 ,69386   ,647,647,647
BEGIN DESCRIPTION:
X18525
END DESCRIPTION:
XS GIS Cut Line= 3
      2495764.86     13835923.34      2495377.35     13834427.78
      2494730.54     13833859.55
#Sta/Elev= 30
  3762.3  425.95  3795.5  424.48  3911.8  421.99  4301.4  411.15  4418.1  410.83
    4587  406.77  4833.3  405.17  4859.4  404.02  4940.6  405.49  4969.2  403.81
  4976.1  402.17  4981.2  403.53  4986.7  396.49  4987.2  395.99  5013.7  396.49
  5016.7  403.95  5021.8  403.18  5092.7  405.89  5229.8  414.23  5323.8  415.84
  5364.5  417.78  5579.7  422.69  5679.5  427.75  5741.4  429.41  5791.5  431.66
  5892.1  434.45  5963.5  438.47  5980.7  438.67  6091.5   445.5  6168.2  447.12
#Mann= 15 ,-1 , 0
  3762.3     .05       0  3795.5     .07       0  3911.8     .05       0
  4833.3      .1       0  4986.7     .05       0  5013.7      .1       0
  5229.8     .05       0  5323.8     .07       0  5364.5     .05       0
  5579.7     .07       0  5741.4    .035       0  5791.5     .07       0
  5963.5     .12       0  5980.7    .035       0  6091.5     .12       0
Bank Sta=4986.7,5013.7
XS Rating Curve= 0 ,0
Exp/Cntr=0.3,0.1

Type RM Length L Ch R = 1 ,68739   ,666,666,666
BEGIN DESCRIPTION:
Cooperas Creek 76.0
END DESCRIPTION:
XS GIS Cut Line= 3
      2497012.17     13835602.42      2496467.25     13834960.61
       2494693.6     13833719.67
#Sta/Elev= 30
  3498.6  434.81  3609.7   430.8    3655  428.73  4261.1  407.34    4390  401.84
  4396.1  404.69    4417  404.79  4425.7  400.59  4440.5  399.36  4461.5  402.47
  4467.6  400.53  4497.2  409.31  4636.6  413.99  4733.8  413.78  4928.8  407.11
  4970.7  401.04    4972  395.82  4972.5  395.32  4999.1  395.82  5000.3  400.85
  5021.3  404.94    5172  404.02  5545.3  410.11    5914  425.47  6035.1   430.5
  6216.8  438.62  6385.5  444.61  6392.8   444.7  6466.1  445.21  6505.2  445.69
#Mann= 14 ,-1 , 0
  3498.6     .05       0  3609.7    .035       0    3655     .07       0
  4261.1     .12       0  4636.6     .07       0    4972     .05       0
  4999.1     .07       0    5172     .05       0    5914     .07       0
  6035.1     .05       0  6216.8    .035       0  6385.5     .12       0
  6392.8    .035       0  6466.1     .05       0
Bank Sta=4972,4999.1
XS Rating Curve= 0 ,0
Exp/Cntr=0.3,0.1

Type RM Length L Ch R = 1 ,68073   ,673,673,673
BEGIN DESCRIPTION:
Cooperas Creek 75.0
END DESCRIPTION:
XS GIS Cut Line= 3
      2497284.68     13835457.15      2496612.57     13834349.06
      2494753.88     13833549.89
#Sta/Elev= 30
  3006.2   436.1  3277.7  429.58  3458.9  420.51  3642.9  420.17  3850.7  415.63
  3874.8  414.89  3976.3  408.26  4056.3  404.45  4237.8  403.88  4301.6  401.49
  4325.9  394.71  4332.2  400.78  4346.7  401.11  4824.5  402.04  4916.7  403.05
  4987.1  401.46  5004.4  394.05  5004.9  393.55  5031.6  394.05  5039.7  399.79
  5057.7  402.65  5154.1  402.91    5301  406.05  5344.5  414.56  5385.5   409.2
  5443.5  409.12  5994.1  435.31  6203.9  440.58  6234.2  440.32  6325.4  440.84
#Mann= 15 ,-1 , 0
  3006.2     .05       0  3642.9     .07       0  3850.7     .05       0
  3874.8    .035       0  3976.3     .05       0  4056.3    .035       0
  4237.8      .1       0  4346.7     .05       0  4824.5     .07       0
  4916.7      .1       0  5004.4     .05       0  5031.6      .1       0
  5154.1     .05       0  6203.9    .035       0  6234.2     .05       0
Bank Sta=5004.4,5031.6
XS Rating Curve= 0 ,0
Exp/Cntr=0.3,0.1

Type RM Length L Ch R = 1 ,67400   ,1315,1315,1315
BEGIN DESCRIPTION:
Cooperas Creek 74.0
END DESCRIPTION:
XS GIS Cut Line= 3
      2497363.39     13835299.71      2496122.11     13833398.43
      2494869.34     13833295.55
#Sta/Elev= 30
  2967.4  433.88  3115.2  430.34  3151.4  426.43  3193.5   427.8  3389.7  421.35
  3641.8  420.68  3980.9  403.99    4097  402.53  4269.7  401.49  4327.9  395.88
    4349  400.42  4379.2  401.74  4479.3  401.91  4680.8   400.1  4812.2  403.19
  4970.8  402.15  4985.6  399.21    4993  394.46  4993.5  393.96  5020.2  394.46
  5027.7  399.35  5063.9  404.55  5125.9  408.59  5320.3  413.03  5537.3   412.6
    5705  412.26  5830.9  414.76  6178.3  431.39  6460.2  435.33    6495   435.3
#Mann= 12 ,-1 , 0
  2967.4     .05       0    4097    .035       0  4269.7      .1       0
  4479.3     .05       0  4970.8      .1       0    4993     .05       0
  5020.2      .1       0  5125.9     .07       0  5320.3     .05       0
  5537.3     .07       0    5705     .05       0  6460.2    .035       0
Bank Sta=4993,5020.2
XS Rating Curve= 0 ,0
Exp/Cntr=0.3,0.1

Type RM Length L Ch R = 1 ,66085   ,636,636,636
BEGIN DESCRIPTION:
X18524
END DESCRIPTION:
XS GIS Cut Line= 3
      2498246.49     13834445.36      2496270.31     13833308.38
      2494889.85     13833145.97
#Sta/Elev= 30
  3646.1  426.86  3684.7  425.88    3867  425.42  4122.4  417.89  4234.2  414.15
  4405.5  409.91    4519  406.58  4669.8  406.84  4793.4  403.23  4834.2  402.98
  4951.5   403.6  4986.1  399.51  4995.1  388.93  4995.6  388.43  5023.2  388.93
  5023.5   393.9  5039.2  399.21  5089.9   396.6  5098.2  398.68  5128.9  399.52
  5240.7  398.28  5576.2  402.34  6072.3   410.9  6389.2  411.49  6545.6  411.32
  6744.6  418.14  7024.3  429.76  7198.6  433.41  7297.4  432.63    7316   432.7
#Mann= 17 ,-1 , 0
  3646.1    .035       0  3684.7     .05       0  4122.4    .035       0
  4234.2     .05       0  4405.5     .12       0  4669.8     .07       0
  4793.4    .035       0  4834.2      .1       0  4995.1     .05       0
  5023.2      .1       0  5128.9      .1       0  5240.7    .035       0
  5576.2     .05       0  6389.2     .07       0  6744.6    .035       0
  7198.6     .05       0  7297.4    .035       0
Bank Sta=4995.1,5023.2
XS Rating Curve= 0 ,0
Exp/Cntr=0.3,0.1

Type RM Length L Ch R = 1 ,65449   ,1077,1077,1077
BEGIN DESCRIPTION:
Cooperas Creek 73.0
END DESCRIPTION:
XS GIS Cut Line= 3
      2498639.05     13834120.52        2497225.       13833225.
      2495255.11     13832983.52
#Sta/Elev= 30
  3326.7  419.77  3579.2  416.84  3687.6  414.82  4449.6  403.31  4798.4  402.62
  4883.5  400.51  4935.2  401.16  4977.6  397.21  4983.5     388    4984   387.5
  5011.6     388  5015.2  391.28  5020.6   396.2  5030.7  398.51  5060.9  397.27
  5091.1  399.23  5152.7  398.79  5251.6  397.35  5450.6  400.01  5514.3  397.19
  5548.3  398.21  5647.2  399.67  5746.1  400.64    5944  404.76  6141.8  406.59
  6636.3  410.42  6723.3  411.99  6898.9  418.75  6955.3  421.38  6985.1  422.55
#Mann= 16 ,-1 , 0
  3326.7     .12       0  3579.2     .07       0  3687.6     .05       0
  4798.4      .1       0  4983.5     .05       0  5011.6      .1       0
  5015.2     .07       0  5152.7     .05       0  5251.6    .035       0
  5548.3     .05       0  5647.2    .035       0  5746.1     .05       0
  6141.8    .035       0  6636.3     .05       0  6898.9    .035       0
  6955.3     .05       0
Bank Sta=4983.5,5011.6
XS Rating Curve= 0 ,0
Exp/Cntr=0.3,0.1

Type RM Length L Ch R = 1 ,64372   ,543,543,543
BEGIN DESCRIPTION:
Cooperas Creek 72.0
END DESCRIPTION:
XS GIS Cut Line= 3
      2499275.04     13833625.02        2496875.       13832625.
      2495349.98      13832672.2
#Sta/Elev= 30
  2395.3  418.87  2420.9  417.82  2444.2  417.92  2634.9  413.35  2950.2  408.69
  3466.5  405.66  3517.4   404.8  3819.4  402.23  4179.8  399.89  4366.6  399.12
    4490  401.29  4629.8   398.9  4803.1  396.26  4894.9  398.26  4962.8  398.55
  4973.7  396.39  4980.7     391  4986.1  394.19  4991.3  388.02  4991.8  387.52
  5019.4  388.02  5025.4  392.45  5035.4  395.38  5075.6   395.4  5095.4  398.17
  5211.2  397.48  5545.6  398.71  6005.8  407.98  6185.9  407.01  6521.1  411.89
#Mann= 16 ,-1 , 0
  2395.3     .05       0  2420.9     .07       0  2444.2     .05       0
  2634.9     .12       0  2950.2     .07       0  3466.5     .12       0
  3517.4     .07       0  3819.4     .05       0  4179.8     .07       0
  4366.6     .05       0  4629.8     .12       0  4894.9      .1       0
  4991.3     .05       0  5019.4      .1       0  5075.6     .07       0
  5211.2     .05       0
Bank Sta=4991.3,5019.4
XS Rating Curve= 0 ,0
Exp/Cntr=0.3,0.1

Type RM Length L Ch R = 1 ,63829   ,532,532,532
BEGIN DESCRIPTION:
Cooperas Creek 71.0
END DESCRIPTION:
XS GIS Cut Line= 3
      2499025.02     13833375.01        2496625.       13832175.
      2496374.99     13831724.98
#Sta/Elev= 30
  2316.7  415.87  2369.4  413.67  2473.2  410.51  2783.5  407.27  2934.4  406.35
  2995.9  403.87  3058.5  404.89  3346.1  402.57    3516  401.05  3712.7  400.02
  3821.3  399.67  4233.3  399.04  4404.6  399.97  4561.1  395.99    4679  396.51
  4812.7  397.51  4851.9  394.37  4879.8  396.91  4932.9  395.57  4969.3  392.53
    4971  385.94  4971.5  385.44    5001  385.94    5008   389.2  5013.7  394.48
  5022.9  396.15  5137.4  397.76  5242.2  402.48  5356.5  406.78  5514.8  413.71
#Mann= 16 ,-1 , 0
  2316.7    .035       0  2369.4     .12       0  2783.5     .07       0
  3058.5     .12       0  3346.1     .07       0    3516     .05       0
  3712.7     .07       0  3821.3     .05       0  4233.3     .12       0
  4561.1    .035       0    4679      .1       0    4971     .05       0
    5001      .1       0  5137.4     .05       0  5242.2     .07       0
  5356.5     .05       0
Bank Sta=4971,5001
XS Rating Curve= 0 ,0
Exp/Cntr=0.3,0.1

Type RM Length L Ch R = 1 ,63297   ,576,576,576
BEGIN DESCRIPTION:
Cooperas Creek 70.0
END DESCRIPTION:
XS GIS Cut Line= 3
      2499175.02     13833225.01        2496975.       13831825.
      2496324.99       13831675.
#Sta/Elev= 30
  2392.8  432.48  2403.7  432.04  2436.9  428.45  2545.8  422.42    2552  423.29
  2624.8  418.26  2771.4  412.56  2853.5  410.56  2932.5  408.64    3198  402.61
  3391.9  402.71  3449.4  400.83  3464.7  401.92    3513  398.88  3616.2  400.34
  3881.9  398.65  4016.5   397.7  4695.7  396.74  4804.6  394.26  4862.5  393.07
  4964.9  398.06  4992.9   394.4  4995.8  384.81  4996.3  384.31  5025.8  384.81
  5031.3  394.14  5228.4  397.39  5390.5   402.1    5565  412.39  5667.6  416.41
#Mann= 13 ,-1 , 0
  2392.8     .07       0  2403.7     .05       0  2545.8    .035       0
  2771.4     .12       0  2853.5     .05       0  2932.5     .12       0
    3513     .05       0  3881.9     .07       0  4016.5     .05       0
  4804.6      .1       0  4995.8     .05       0  5025.8      .1       0
  5228.4     .05       0
Bank Sta=4995.8,5025.8
XS Rating Curve= 0 ,0
Exp/Cntr=0.3,0.1

Type RM Length L Ch R = 1 ,62721   ,1028,1028,1028
BEGIN DESCRIPTION:
Cooperas Creek 69.0
END DESCRIPTION:
XS GIS Cut Line= 3
        2499375.       13833325.        2497175.       13831325.
      2496424.97       13831375.
#Sta/Elev= 30
  2026.4  440.49  2077.3  443.56  2139.6  443.82  2466.7  422.48  2481.6  420.91
  2824.1  408.03  2917.4  405.74  2985.9  404.15  3151.9  401.09  3236.5  400.47
  3243.9  400.39  3706.2  396.77  3814.5  396.57  4207.1  394.89  4293.3  394.32
  4312.7  394.23  4326.9  389.84  4355.3  395.49  4455.7   394.7  4575.8  393.44
  4631.7  390.58    4929  395.89  5029.7  391.91  5039.7  390.24  5044.7  383.61
  5045.2  383.11  5074.8  383.61  5109.9  394.74  5213.8   392.8  5751.3  410.73
#Mann= 19 ,-1 , 0
  2026.4     .07       0  2077.3     .05       0  2466.7    .035       0
  2481.6     .05       0  2824.1    .035       0  2917.4     .05       0
  2985.9    .035       0  3151.9     .12       0  3236.5    .035       0
  3243.9     .05       0  3706.2     .07       0  3814.5     .05       0
  4207.1     .07       0  4293.3      .1       0  4455.7     .07       0
  4575.8      .1       0  5044.7     .05       0  5074.8      .1       0
  5213.8     .05       0
Bank Sta=5044.7,5074.8
XS Rating Curve= 0 ,0
Exp/Cntr=0.3,0.1

Type RM Length L Ch R = 1 ,61693   ,534,534,534
BEGIN DESCRIPTION:
Cooperas Creek 68.0
END DESCRIPTION:
XS GIS Cut Line= 3
      2499275.03     13833125.03        2497725.       13831575.
        2497525.       13829175.
#Sta/Elev= 30
    2813  440.65  3095.9     420  3669.3  401.65  3673.9  401.44  3769.5  400.09
  3888.2  399.02  4126.5  396.35  4374.2  395.42  4753.1  396.07  4888.6   395.3
  4962.7  393.37  4975.8  383.34  4976.3  382.84    5006  383.34  5025.1  391.53
  5075.3  393.94  5458.3   393.7    5640  391.25  5965.5  395.86  6064.5  395.64
  6199.2  395.22  6249.4  389.77  6309.6  394.48  6379.8   389.2  6460.3  395.17
  6670.1  402.03  6856.2  414.28  7178.2  446.97  7252.1  453.28  7413.4  459.73
#Mann= 20 ,-1 , 0
    2813     .05       0  3669.3    .035       0  3673.9     .05       0
  3769.5    .035       0  3888.2     .05       0  4126.5     .07       0
  4374.2     .05       0  4753.1     .07       0  4888.6      .1       0
  4975.8     .05       0    5006      .1       0  5458.3     .07       0
    5640     .05       0  5965.5     .07       0  6064.5      .1       0
  6460.3     .05       0  6670.1    .035       0  6856.2     .07       0
  7178.2     .12       0  7252.1     .07       0
Bank Sta=4975.8,5006
XS Rating Curve= 0 ,0
Exp/Cntr=0.3,0.1

Type RM Length L Ch R = 1 ,61159   ,540,540,540
BEGIN DESCRIPTION:
Cooperas Creek 67.0
END DESCRIPTION:
XS GIS Cut Line= 3
      2499425.03     13832725.03        2498025.       13831175.
      2497625.01     13829575.05
#Sta/Elev= 30
  2911.5  433.06    3121  417.88  3322.2   405.1  3591.2  397.97  4440.3  394.86
    4689  391.74  4724.1  390.53  4730.8  387.99  4780.9   392.8  4907.9  389.92
    4958  392.81  4972.2  392.05    4978  381.58  4978.5  381.08  5008.2  381.58
  5023.4  387.66  5064.6  393.42  5299.6  390.62  5465.2  394.79  5722.7   394.7
  5866.1  393.63  5907.3  387.55  5917.6  392.77  6078.1  394.48  6268.1  398.92
  6351.8  404.53  6486.7  415.65    6567  423.04    6585  427.16  6649.4   429.6
#Mann= 11 ,-1 , 0
  2911.5     .07       0    3121     .05       0  4440.3      .1       0
    4978     .05       0  5008.2      .1       0  5299.6     .07       0
  5465.2     .05       0  5722.7      .1       0  6078.1     .05       0
  6351.8    .035       0  6486.7     .07       0
Bank Sta=4978,5008.2
XS Rating Curve= 0 ,0
Exp/Cntr=0.3,0.1

Type RM Length L Ch R = 1 ,60619   ,566,566,566
BEGIN DESCRIPTION:
Cooperas Creek 66.0
END DESCRIPTION:
XS GIS Cut Line= 3
      2499974.98     13832374.98        2498425.       13830825.
      2497574.99     13829224.98
#Sta/Elev= 30
    2808  420.02  2971.9  409.62  3107.4   402.3  3297.5  397.68    4051  392.99
  4400.1  393.16  4696.5  392.07  4733.2  391.46  4985.9  390.25  4996.5  388.17
  4998.5  381.45    4999  380.95  5029.1  381.45  5030.1  388.06  5067.9  391.85
  5304.6  393.14  5332.2  384.42  5452.8  391.24  5458.4  384.81  5474.8  389.55
  5496.7  384.73  5650.6  392.04  5747.4  386.36  5778.3  393.38  6056.6  398.18
  6401.6  428.53    6601  445.77  6683.3   451.5  6800.3  458.78  6811.8  459.07
#Mann= 16 ,-1 , 0
    2808     .07       0  2971.9     .05       0  3107.4     .12       0
  3297.5    .035       0    4051     .05       0  4400.1    .035       0
  4696.5     .05       0  4733.2      .1       0  4998.5     .05       0
  5029.1      .1       0  5778.3     .05       0  6056.6     .07       0
  6401.6    .035       0    6601     .07       0  6683.3    .035       0
  6800.3     .07       0
Bank Sta=4998.5,5029.1
XS Rating Curve= 0 ,0
Exp/Cntr=0.3,0.1

Type RM Length L Ch R = 1 ,60053   ,569,569,569
BEGIN DESCRIPTION:
Cooperas Creek 65.0
END DESCRIPTION:
XS GIS Cut Line= 3
      2500475.01     13831975.01        2498925.       13830725.
        2497625.     13829124.99
#Sta/Elev= 30
  3004.2  448.86  3132.7  439.07  3444.9  407.04  3679.9   395.2  3759.5  394.84
  3796.9  394.15  4169.3  391.35  4252.4  391.12  4300.3  390.86  4386.4  390.85
  4477.9  391.04  4676.1  391.51  4787.6  391.91  4959.5  391.52  4981.8  389.33
  4986.4  380.02  4986.9  379.52  5018.9  380.02  5023.4  389.66  5045.7  391.66
  5196.5  390.24  5901.2  391.74  6090.6  394.37  6302.1  408.94  6515.4  423.83
  6628.5  434.54  6818.7  449.61  6905.6   454.7  6969.7  457.89    7057  460.09
#Mann= 20 ,-1 , 0
  3004.2     .12       0  3759.5    .035       0  3796.9     .05       0
  4169.3    .035       0  4252.4     .05       0  4300.3    .035       0
  4386.4     .05       0  4477.9    .035       0  4676.1     .05       0
  4787.6      .1       0  4986.4     .05       0  5018.9      .1       0
  5196.5    .035       0  5901.2     .05       0  6302.1     .07       0
  6515.4     .05       0  6628.5     .07       0  6818.7    .035       0
  6905.6     .05       0  6969.7    .035       0
Bank Sta=4986.4,5018.9
XS Rating Curve= 0 ,0
Exp/Cntr=0.3,0.1
