HEC-RAS study DENTON CREEK 2.prj: DENTON CREEK 2 Base Level Engineering

--- DENTON CREEK 2.g01 (geometry) --- (continued)

Type RM Length L Ch R = 1 ,61297   ,477,477,477
BEGIN DESCRIPTION:
DENTON CREEK 2 68.0
END DESCRIPTION:
XS GIS Cut Line= 3
      2480124.97     13762374.98        2479525.       13761825.
      2479074.99     13761324.99
#Sta/Elev= 30
  4186.6  326.72  4353.5  325.36  4490.9  324.12  4618.5  324.25  4661.1  322.71
    4682  323.13  4905.4  319.16  4950.9  319.11    4965  313.85  4972.4  308.71
  4978.1  306.17  4978.6  305.67  4995.1  306.17  4997.1   310.5  5007.6  311.32
  5028.5  311.87  5078.6   310.6  5148.9  311.74  5170.5  310.98  5227.3  312.45
  5297.6  311.04    5326  313.36  5347.7  317.01  5368.6  318.65  5400.8  319.03
  5482.2   321.4  5517.3  325.26  5545.7  325.85  5637.7  331.52  5673.2  332.47
#Mann= 6 ,-1 , 0
  4186.6     .05       0  4353.5     .07       0  4905.4      .1       0
  4978.1     .05       0  4995.1      .1       0  5400.8     .12       0
Bank Sta=4978.1,4995.1
XS Rating Curve= 0 ,0
Exp/Cntr=0.3,0.1

Type RM Length L Ch R = 1 ,60820   ,466,466,466
BEGIN DESCRIPTION:
DENTON CREEK 2 67.0
END DESCRIPTION:
XS GIS Cut Line= 3
      2480324.99     13762024.99        2479725.       13761425.
      2479124.98       13761275.
#Sta/Elev= 30
  4147.5  326.46  4204.1  325.37  4303.1  321.63  4334.4  322.88  4373.8  321.54
  4444.5  322.72  4479.5  321.94  4722.4  318.07    4798  315.36  4826.3  312.52
  4840.5  309.85  4865.7  312.02  4882.9  311.97    4897  314.21  4911.2  314.45
  4925.3  311.92  4939.4  310.78  4967.7  311.07  4983.8  306.29  4984.3  305.79
  5001.1  306.29  5037.2  311.25  5047.6  311.58    5130  310.65  5181.4  311.83
  5233.1  314.27  5417.8  317.66  5472.7   319.6  5562.9   327.9  5614.5  329.98
#Mann= 10 ,-1 , 0
  4147.5     .05       0  4303.1     .07       0  4334.4     .12       0
  4479.5     .07       0  4722.4     .12       0  4865.7      .1       0
  4983.8     .05       0  5001.1      .1       0  5181.4     .07       0
  5417.8     .12       0
Bank Sta=4983.8,5001.1
XS Rating Curve= 0 ,0
Exp/Cntr=0.3,0.1

Type RM Length L Ch R = 1 ,60354   ,931,931,931
BEGIN DESCRIPTION:
DENTON CREEK 2 66.0
END DESCRIPTION:
XS GIS Cut Line= 3
      2480825.02     13760724.99        2479625.       13761025.
      2479174.99       13761175.
#Sta/Elev= 30
  3767.4  339.84  3939.6  331.31  4128.2  324.55  4244.2  322.25  4272.5  323.05
  4293.1  319.61  4326.6  321.69  4467.3  320.05  4651.3  318.05  4684.8  313.51
  4715.7  313.43  4733.8  311.46  4738.9  313.64    4757  313.64    4775  311.45
  4780.2  312.94  4816.2  307.18  4821.4  308.89  4945.1   310.1  4963.1  309.11
  4972.5   303.5    4973     303  4989.8   303.5    4994  303.59  5001.8  309.03
  5040.5  315.14  5130.8  315.82  5324.4  320.61  5404.9  322.82  5478.7  327.19
#Mann= 7 ,-1 , 0
  3767.4     .07       0  3939.6     .05       0  4467.3      .1       0
  4972.5     .05       0  4989.8      .1       0  5040.5     .07       0
  5324.4     .12       0
Bank Sta=4972.5,4989.8
XS Rating Curve= 0 ,0
Exp/Cntr=0.3,0.1

Type RM Length L Ch R = 1 ,59423   ,465,465,465
BEGIN DESCRIPTION:
DENTON CREEK 2 65.0
END DESCRIPTION:
XS GIS Cut Line= 3
      2480675.02       13760375.        2479775.       13760275.
      2478875.01     13761274.98
#Sta/Elev= 30
  4089.8  336.62  4230.7   330.3  4361.5  322.29    4613   317.8  4734.7  317.16
  4804.2  316.51  4814.3   313.9  4824.3  313.47  4833.5  315.64  4884.7  317.08
  4914.9  313.83  4945.1   307.2  4975.2  308.49  4998.7  307.74  5000.5  302.75
    5001  302.25  5017.9  302.75  5023.4  303.33  5030.9   307.3  5051.8  308.45
  5073.7  305.81  5087.7  305.03  5101.9  307.87  5214.7  313.12  5629.5  319.82
  5839.8  322.15  5962.2  325.71  5975.6  326.19  6213.3  335.96  6340.7  339.52
#Mann= 10 ,-1 , 0
  4089.8     .05       0  4734.7      .1       0  4833.5    .035       0
  5000.5    .035       0  5017.9    .035       0  5073.7     .07       0
  5629.5     .05       0  5839.8     .07       0  5962.2     .12       0
  5975.6     .07       0
Bank Sta=5000.5,5017.9
XS Rating Curve= 0 ,0
Exp/Cntr=0.3,0.1

Type RM Length L Ch R = 1 ,58958   ,915,915,915
BEGIN DESCRIPTION:
DENTON CREEK 2 64.0
END DESCRIPTION:
XS GIS Cut Line= 3
        2480575.       13760275.        2479675.       13759875.
      2478574.99       13760375.
#Sta/Elev= 30
  4016.1   331.5  4198.7  321.69  4317.1  320.36    4387  317.46  4401.2  319.11
  4424.4  319.35  4572.9  317.72  4592.7  316.46    4772  314.99  4893.6  312.74
  4916.9  311.22  4934.6  307.54  4957.2  306.35  4963.4  304.66  4968.8   305.8
  4979.1  305.43  4986.6  302.42  4992.1  304.78    5001   301.8  5001.5   301.3
  5018.5   301.8    5023   306.9  5114.4  307.94  5143.8  309.93    5280  311.85
  5407.4  317.09  5566.2  319.15  5790.1  320.76    6005  323.76  6209.3  332.12
#Mann= 10 ,-1 , 0
  4016.1     .05       0  4317.1    .035       0    4387     .05       0
  4572.9     .07       0    4772      .1       0    5001     .05       0
  5018.5      .1       0  5114.4     .07       0  5566.2    .035       0
  5790.1     .07       0
Bank Sta=5001,5018.5
XS Rating Curve= 0 ,0
Exp/Cntr=0.3,0.1

Type RM Length L Ch R = 1 ,58043   ,1249,1249,1249
BEGIN DESCRIPTION:
DENTON CREEK 2 63.0
END DESCRIPTION:
XS GIS Cut Line= 3
        2480775.       13760375.        2479675.       13759175.
        2479675.     13758974.98
#Sta/Elev= 30
  3375.9  340.29  3496.4  337.67  3666.6   329.3  3803.8  324.13  3814.6  324.09
  3828.8  320.33  3850.4  323.53    3999  322.05  4040.9  319.27  4749.3  307.52
  4812.9  304.58    4869     305  4876.4  303.54  4883.2  305.17  4890.6  301.53
  4897.4  303.92  4904.8  302.45    4919  305.33    4940  305.95  4961.5   303.7
  4966.9  298.79  4967.4  298.29  4984.5  298.79  4989.9  303.85  5000.4   307.9
  5006.3   307.9  5023.8  315.31  5125.3  320.19  5127.1  320.18  5203.8  322.64
#Mann= 8 ,-1 , 0
  3375.9     .05       0  3666.6    .035       0  3803.8     .05       0
  4749.3      .1       0  4966.9     .05       0  4984.5      .1       0
  5125.3     .07       0  5127.1     .12       0
Bank Sta=4966.9,4984.5
XS Rating Curve= 0 ,0
Exp/Cntr=0.3,0.1

Type RM Length L Ch R = 1 ,56794   ,1361,1361,1361
BEGIN DESCRIPTION:
DENTON CREEK 2 62.0
END DESCRIPTION:
XS GIS Cut Line= 3
      2480925.01     13759575.01        2480325.       13759075.
      2479774.95     13758974.99
#Sta/Elev= 30
  4214.6  341.78  4217.9  341.78  4221.8  340.56  4242.6   339.7    4279  336.38
  4299.9  332.58  4328.5  329.28  4390.3  324.62  4519.9  315.95  4722.4  310.59
    4775  309.79    4818  308.02  4839.4  307.96  4846.6  308.63  4881.7  306.99
  4896.1   303.8  4903.9  303.42  4998.2   303.6  5007.1  296.22  5007.6  295.72
  5024.8  296.22  5027.4  299.08  5036.3  302.98  5056.6  306.51  5066.8  307.26
  5117.6  307.42  5142.5  308.38  5290.4  312.68  5482.5  315.42  5554.7   318.8
#Mann= 7 ,-1 , 0
  4214.6     .12       0  4390.3     .05       0  4722.4      .1       0
  5007.1     .05       0  5024.8      .1       0  5142.5     .05       0
  5482.5     .12       0
Bank Sta=5007.1,5024.8
XS Rating Curve= 0 ,0
Exp/Cntr=0.3,0.1

Type RM Length L Ch R = 1 ,55433   ,450,450,450
BEGIN DESCRIPTION:
DENTON CREEK 2 61.0
END DESCRIPTION:
XS GIS Cut Line= 3
      2481124.98       13758475.        2480875.       13758425.
      2479775.03     13758924.99
#Sta/Elev= 30
  4740.5  326.83  4781.3  326.22  4791.5  324.68  4795.6   323.1  4811.9   317.3
  4832.3  311.62  4842.5  306.73  4852.7  303.95  4895.5  301.43  4903.6  301.45
  4913.8  299.46  4944.4  302.01  4998.2   300.8  5000.8  295.38  5001.3  294.88
  5018.6  295.38  5027.3  301.22  5039.4  303.43  5085.3  303.04  5228.3   306.8
  5357.9  306.72  5585.3  308.37  5706.1  307.75  5797.3  310.73  5907.2  312.85
    6039  313.54  6139.6   315.5  6159.8   316.3  6166.4  317.29  6203.7  318.32
#Mann= 7 ,-1 , 0
  4740.5     .07       0  4795.6     .12       0  4895.5      .1       0
  5000.8     .05       0  5018.6      .1       0  5085.3     .05       0
  6139.6     .12       0
Bank Sta=5000.8,5018.6
XS Rating Curve= 0 ,0
Exp/Cntr=0.3,0.1

Type RM Length L Ch R = 1 ,54983   ,429,429,429
BEGIN DESCRIPTION:
DENTON CREEK 2 60.0
END DESCRIPTION:
XS GIS Cut Line= 3
      2481174.99       13757975.        2480575.       13758175.
      2479675.01     13758874.99
#Sta/Elev= 30
  4371.4  328.08  4424.1  321.35  4508.4  314.25  4583.5  305.76  4624.4  304.89
  4645.5  306.63    4656  304.28  4705.5  305.09    4793  303.92  4803.6  302.07
  4824.6   302.3  4835.2  299.72  4856.3  301.24  4887.9  301.11    4909  298.05
  4910.6  296.59  4911.1  296.09  4928.5  296.59  4930.1  301.29  4979.9  301.37
  4993.3   299.7  5001.2  296.73    5007  296.73    5040  303.72  5067.2  306.41
  5338.7  307.73  5452.7  306.62    5967  315.25  6058.1  318.21    6144  323.43
#Mann= 7 ,-1 , 0
  4371.4     .07       0  4583.5     .05       0  4705.5      .1       0
  4910.6     .05       0  4928.5      .1       0  4979.9     .05       0
    5967     .12       0
Bank Sta=4910.6,4928.5
XS Rating Curve= 0 ,0
Exp/Cntr=0.3,0.1

Type RM Length L Ch R = 1 ,54554   ,1751,1751,1751
BEGIN DESCRIPTION:
DENTON CREEK 2 59.0
END DESCRIPTION:
XS GIS Cut Line= 3
      2480975.02       13757775.        2480725.       13757825.
      2479824.96     13758225.02
#Sta/Elev= 30
  4739.8  327.39  4778.3  320.91  4811.2   310.2  4831.6   306.4  4913.2  303.95
  4970.8  305.43  4984.6   304.7  4992.2   300.2  4997.5   300.2  5003.7  293.85
  5009.1  297.88  5016.7  292.09  5026.9  294.96  5032.4   292.3  5038.5  295.89
  5049.5  296.85  5052.2  292.02  5052.7  291.52  5070.1  292.02  5084.4  297.78
  5102.1  293.31  5130.9  293.88  5154.1  298.36  5159.6  295.32  5169.9  297.87
  5177.4  303.14  5182.9  298.04  5191.7  302.56  5213.3  302.94  5979.7  312.56
#Mann= 6 ,-1 , 0
  4739.8     .07       0  4778.3     .05       0  4970.8      .1       0
  5052.2     .05       0  5070.1      .1       0  5213.3     .05       0
Bank Sta=5052.2,5070.1
XS Rating Curve= 0 ,0
Exp/Cntr=0.3,0.1

Type RM Length L Ch R = 1 ,52803   ,448,448,448
BEGIN DESCRIPTION:
DENTON CREEK 2 58.0
END DESCRIPTION:
XS GIS Cut Line= 3
      2480925.01       13757625.        2480025.       13757325.
      2479424.99       13757325.
#Sta/Elev= 30
  4051.3  321.72  4062.3   322.1  4072.4  323.18  4114.6  313.09  4167.3  306.97
    4220  304.32    4277   303.3  4367.5  309.19  4409.7   308.6  4475.7  305.29
  4604.7   304.5    4610  305.63  4631.1  303.73  4641.6   305.2  4652.1  304.29
  4673.2  306.04  4683.8  304.32  4778.6   301.1  4877.5  299.94  4957.8  299.15
  4978.9  296.52  4987.4  290.75  4987.9  290.25  5007.4  290.75    5010  292.82
    5020  296.47    5070  297.79  5103.3  302.31  5424.4  307.59    5600  310.51
#Mann= 9 ,-1 , 0
  4051.3     .07       0  4062.3     .05       0    4277      .1       0
  4475.7     .05       0  4877.5      .1       0  4987.4     .05       0
  5007.4      .1       0  5103.3     .07       0  5424.4     .05       0
Bank Sta=4987.4,5007.4
XS Rating Curve= 0 ,0
Exp/Cntr=0.3,0.1

Type RM Length L Ch R = 1 ,52355   ,1099,1099,1099
BEGIN DESCRIPTION:
DENTON CREEK 2 57.0
END DESCRIPTION:
XS GIS Cut Line= 3
      2481174.98     13757724.99        2480075.       13756925.
      2479475.04     13757224.98
#Sta/Elev= 30
  3635.6  330.25  3727.9  329.45  3793.6  329.36  3858.1  327.05  3900.3  323.99
  3965.2  316.31  3979.9   316.6  4000.7  313.55  4065.6  308.35    4187  303.98
  4213.4  304.67  4243.4  303.96  4272.8   301.5  4408.8  304.76  4833.1  303.21
  4938.2   302.6  4952.8  298.43    4959   299.6  4967.5  296.16  4973.7  296.93
  4982.2  293.25  4998.5  293.08  4999.7  289.11  5000.2  288.61  5019.7  289.11
  5026.5  296.37  5151.9  298.88  5227.7  299.77  5479.3  307.23  5666.5  309.42
#Mann= 7 ,-1 , 0
  3635.6     .05       0  3727.9     .07       0  4213.4     .05       0
  4833.1      .1       0  4999.7     .05       0  5019.7      .1       0
  5151.9     .05       0
Bank Sta=4999.7,5019.7
XS Rating Curve= 0 ,0
Exp/Cntr=0.3,0.1

Type RM Length L Ch R = 1 ,51256   ,1065,1065,1065
BEGIN DESCRIPTION:
DENTON CREEK 2 56.0
END DESCRIPTION:
XS GIS Cut Line= 4
      2481437.31     13757053.56      2479676.02     13756176.02
        2479625.       13756125.        2478925.       13755475.
#Sta/Elev= 30
  2959.5  321.41    3487  310.86  3535.9  308.77  3594.3  301.95  3666.6  299.98
  3728.6  302.55    3839  302.03  3898.5  301.64  4173.8  299.31  4235.7  298.09
  4325.1  301.33  4403.7  299.26  4512.2  296.82  4584.8  299.53  4729.2  299.33
  4899.2  297.78    4957  295.63  4973.2  289.97  4973.7  289.47  4997.5  289.97
  5013.4  294.96  5091.6  294.46  5105.7  292.39    5185  294.97  5197.6  292.97
  5211.8  295.67  5388.6  301.63  5586.5  304.97  5933.4  316.34  5954.7  316.96
#Mann= 15 ,-1 , 0
  2959.5     .05       0    3487     .12       0  3535.9    .035       0
  3666.6     .12       0    3839     .07       0  3898.5     .12       0
  4173.8     .07       0  4403.7     .12       0  4512.2     .07       0
  4729.2     .05       0  4899.2      .1       0  4973.2     .05       0
  4997.5      .1       0    5185     .05       0  5933.4     .12       0
Bank Sta=4973.2,4997.5
XS Rating Curve= 0 ,0
Exp/Cntr=0.3,0.1

Type RM Length L Ch R = 1 ,50191   ,534,534,534
BEGIN DESCRIPTION:
DENTON CREEK 2 55.0
END DESCRIPTION:
XS GIS Cut Line= 3
      2480924.99     13756574.99        2479675.       13755475.
      2479225.04     13755225.02
#Sta/Elev= 30
  3338.7  311.32  3390.6  310.48  3466.3  306.34  3558.3  310.76  3571.8  308.93
  3607.7  307.84  3615.2  305.47  3636.1  306.66  3643.7  304.27  3650.4  305.43
  3678.8  301.75  3719.1  301.66  3719.8   301.6  3770.9  303.96  3919.8  300.95
    4436  297.65  4597.6     297  4730.5   295.1  4982.4   293.4    4990  292.54
  4999.6  284.45  5000.1  283.95    5024  284.45  5033.5  293.83  5129.6  293.21
  5201.7  302.09  5217.7  300.12  5268.6  303.59  5421.8  308.31  5518.5  313.12
#Mann= 12 ,-1 , 0
  3338.7     .07       0  3390.6    .035       0  3571.8     .12       0
  3719.1     .07       0  3719.8     .05       0    4436     .07       0
  4597.6     .12       0  4730.5      .1       0  4999.6     .05       0
    5024      .1       0  5268.6     .05       0  5421.8     .07       0
Bank Sta=4999.6,5024
XS Rating Curve= 0 ,0
Exp/Cntr=0.3,0.1

Type RM Length L Ch R = 1 ,49657   ,557,557,557
BEGIN DESCRIPTION:
DENTON CREEK 2 54.0
END DESCRIPTION:
XS GIS Cut Line= 3
      2481025.03     13756025.02        2480075.       13755375.
      2479424.99     13754624.99
#Sta/Elev= 30
  3844.6  309.07  4225.8   299.7    4761  296.74    4910   295.4  4995.1  294.09
    4999  294.09  5002.8  289.87  5004.9  283.41  5005.4  282.91  5029.3  283.41
  5031.3  289.14    5038  292.34  5109.2   290.8  5406.1  296.23  5428.3  290.84
  5455.9  291.29  5477.7  296.81  5541.3  298.79  5591.2  298.49  5604.9  295.22
  5633.4  296.14  5641.1  298.87  5647.7  295.43  5661.9  296.91  5683.8  305.32
  5734.1  309.41  5825.3  315.87  5868.3  322.32  5938.3  330.39  5988.2  331.49
#Mann= 10 ,-1 , 0
  3844.6     .05       0    4761     .07       0    4910     .05       0
  4995.1      .1       0  5004.9     .05       0  5029.3      .1       0
  5406.1     .05       0  5455.9     .07       0  5734.1     .05       0
  5868.3     .12       0
Bank Sta=5004.9,5029.3
XS Rating Curve= 0 ,0
Exp/Cntr=0.3,0.1

Type RM Length L Ch R = 1 ,49100   ,551,551,551
BEGIN DESCRIPTION:
DENTON CREEK 2 53.0
END DESCRIPTION:
XS GIS Cut Line= 3
      2481174.98     13755874.98        2480225.       13754925.
      2479475.04     13754625.02
#Sta/Elev= 30
  3656.8  309.96  3859.6  306.42  3965.6  302.71    3991  301.62  4109.3  297.77
  4196.3  297.16  4519.4  298.91  4664.2  296.97  4691.8  296.58    4774  293.76
  4802.3  291.25  4844.7  293.67    4972  293.47    5003   290.7  5009.6  282.17
  5010.1  281.67  5034.1  282.17  5039.3  290.11  5044.7  291.22  5093.2  290.93
  5122.8  293.68  5184.6  294.71  5225.1  293.27  5355.5  298.63  5499.7  304.41
  5624.9  311.86  5732.7  320.62    5769  324.94    5775  326.96    5808  330.91
#Mann= 12 ,-1 , 0
  3656.8     .05       0  3859.6    .035       0  3965.6     .05       0
    3991     .07       0  4196.3     .05       0  4664.2     .07       0
  4691.8      .1       0  5009.6     .05       0  5034.1      .1       0
  5184.6     .07       0  5355.5     .05       0    5775     .12       0
Bank Sta=5009.6,5034.1
XS Rating Curve= 0 ,0
Exp/Cntr=0.3,0.1

Type RM Length L Ch R = 1 ,48549   ,543,543,543
BEGIN DESCRIPTION:
DENTON CREEK 2 52.0
END DESCRIPTION:
XS GIS Cut Line= 3
      2481225.01     13755825.01        2480575.       13754725.
      2480075.01     13754175.01
#Sta/Elev= 30
    3707  309.87  3951.3  306.03    4040  303.49  4145.2  299.28  4275.1  297.73
  4610.4  297.09  4715.5  297.36  4866.9  292.51  4912.6  289.92  4988.1  291.26
  4998.6  284.03    5006  282.73  5012.7  283.09  5026.9  290.61  5034.4  288.71
  5041.1  290.57  5069.5  284.15  5091.1   282.5  5097.9  288.34  5107.3  282.14
  5107.8  281.64  5131.8  282.14  5133.4  287.18  5154.7  295.26    5228  298.67
  5252.2  299.54  5364.5  302.45  5385.6  302.75  5489.9  304.82    5728     313
#Mann= 14 ,-1 , 0
    3707     .05       0  3951.3    .035       0    4040     .05       0
  4145.2     .07       0  4275.1     .05       0  4610.4     .07       0
  4866.9      .1       0  5107.3     .05       0  5131.8      .1       0
    5228     .05       0  5252.2     .07       0  5364.5     .05       0
  5385.6     .07       0  5489.9     .05       0
Bank Sta=5107.3,5131.8
XS Rating Curve= 0 ,0
Exp/Cntr=0.3,0.1

Type RM Length L Ch R = 1 ,48006   ,585,585,585
BEGIN DESCRIPTION:
DENTON CREEK 2 51.0
END DESCRIPTION:
XS GIS Cut Line= 3
      2482224.99     13755924.99        2480975.       13754525.
        2480175.       13754075.
#Sta/Elev= 30
  3128.1  322.42  3304.9  320.47  3361.8  316.34  3404.4  316.33    3447  313.93
  3531.5  313.52  3680.3  309.11  4231.3  303.12  4367.9  301.42    4523  299.31
  4598.4  296.72  4721.9  292.36  4874.3  292.15  4926.8  292.48  4962.7  289.78
  4976.9  290.53  4983.6  287.91  4985.5  285.51    4986  285.01  5010.2  285.51
  5012.9   290.1  5027.9  291.76  5077.9  289.85  5131.1  292.77  5180.5  291.42
  5255.7  293.11  5287.9  295.29  5326.5  298.13  5547.7  301.42  5922.8     311
#Mann= 8 ,-1 , 0
  3128.1     .05       0  4231.3    .035       0  4367.9     .05       0
  4598.4     .07       0  4874.3      .1       0  4985.5     .05       0
  5010.2      .1       0  5287.9     .07       0
Bank Sta=4985.5,5010.2
XS Rating Curve= 0 ,0
Exp/Cntr=0.3,0.1

Type RM Length L Ch R = 1 ,47421   ,516,516,516
BEGIN DESCRIPTION:
DENTON CREEK 2 50.0
END DESCRIPTION:
XS GIS Cut Line= 3
      2482224.98     13755724.96        2481425.       13754175.
        2480625.       13753375.
#Sta/Elev= 30
    3256   320.3  3895.5  304.28  4272.1  300.52  4382.9  297.36  4666.2  295.95
    4704  293.99  4769.7  293.86  4820.4  290.71  4869.7  289.97  4882.1  289.57
  4919.9  291.17  4964.2  290.32  4977.7  287.93  4985.1  282.38  4985.6  281.88
  5009.8  282.38  5014.4  289.57  5128.2  288.44  5169.9  292.52  5254.8  294.25
  5466.9  292.99  5537.6   290.8  5607.9  292.78  5636.6  291.02  5651.9  291.79
  5679.1  297.46  5763.9  297.76  5862.9  301.52  5990.2  303.87  6131.6  309.29
#Mann= 10 ,-1 , 0
    3256     .05       0  4666.2     .12       0  4769.7      .1       0
  4869.7     .12       0  4882.1      .1       0  4985.1     .05       0
  5009.8      .1       0  5128.2     .05       0  5607.9     .12       0
  5651.9     .05       0
Bank Sta=4985.1,5009.8
XS Rating Curve= 0 ,0
Exp/Cntr=0.3,0.1

Type RM Length L Ch R = 1 ,46905   ,571,571,571
BEGIN DESCRIPTION:
DENTON CREEK 2 49.0
END DESCRIPTION:
XS GIS Cut Line= 3
        2482425.     13754975.01        2481775.       13753875.
      2480975.01     13753175.01
#Sta/Elev= 30
  3722.3  310.67  3813.9  308.11  3839.8  307.21  3948.6  303.44  4188.5  297.97
    4638  294.43  4709.4  294.39  4753.6  292.56  4912.2   288.1  4986.4  289.67
  4992.2  288.76  4997.1   285.5  5003.3   285.5  5007.1  287.54  5013.8  281.84
  5023.1  281.59  5023.6  281.09  5048.1  281.59  5049.8  288.37  5056.5   290.4
  5156.4  289.41  5267.6   291.7    5326  292.16  5375.4  293.89    5439  293.62
  5855.1  302.14  5900.2  303.72  5956.7  308.15  6044.9  311.66    6063  312.11
#Mann= 11 ,-1 , 0
  3722.3     .05       0  3813.9     .07       0  3839.8     .05       0
    4638    .035       0  4753.6      .1       0  5023.1     .05       0
  5048.1      .1       0  5156.4     .12       0  5267.6     .05       0
  5855.1     .12       0  6044.9     .07       0
Bank Sta=5023.1,5048.1
XS Rating Curve= 0 ,0
Exp/Cntr=0.3,0.1

Type RM Length L Ch R = 1 ,46334   ,542,542,542
BEGIN DESCRIPTION:
DENTON CREEK 2 48.0
END DESCRIPTION:
XS GIS Cut Line= 3
        2482425.     13754874.97        2482225.       13753625.
      2481524.99     13752874.99
#Sta/Elev= 30
  3733.9  309.43  3822.9  306.81  4027.6  301.59    4220  300.55  4240.2  299.35
  4452.9  296.25  4812.6  292.37    4858   290.8    4939  290.02  4966.2  287.54
    4967  281.59  4967.5  281.09    4992  281.59  4997.2  283.69  5003.2  283.69
  5013.7  289.53    5021  289.82  5035.2  288.65    5106  288.78  5120.2  287.31
  5183.7  286.97  5275.5   289.5  5465.4  292.99  5571.2  296.57  5605.5  297.65
  5701.1  299.76  5813.4  301.74  5919.4  304.95  5997.6  308.53  6025.7   308.8
#Mann= 10 ,-1 , 0
  3733.9     .07       0  3822.9     .05       0  4812.6      .1       0
    4967     .05       0    4992      .1       0  5275.5     .05       0
  5465.4     .07       0  5571.2     .05       0  5605.5     .07       0
  5701.1     .05       0
Bank Sta=4967,4992
XS Rating Curve= 0 ,0
Exp/Cntr=0.3,0.1

Type RM Length L Ch R = 1 ,45792   ,518,518,518
BEGIN DESCRIPTION:
DENTON CREEK 2 47.0
END DESCRIPTION:
XS GIS Cut Line= 3
        2482575.     13754775.04        2482525.       13753225.
        2481925.       13752525.
#Sta/Elev= 30
  3453.7  308.53  3793.9   302.7    3914  302.13  3994.9  299.78  4294.2  293.21
  4314.2  291.53  4524.3  292.74  4644.4  288.35  4805.5  288.78  4924.5  288.39
  4934.5  285.94  4974.5  282.75    4982  280.67  4982.5  280.17  5007.1  280.67
  5007.8  286.76  5011.7  287.87  5018.3  286.93  5025.9  288.16  5032.5  286.05
  5042.1   287.4  5061.1   286.3  5153.3  292.32  5252.4  295.76  5285.3  296.34
  5436.8  297.55  5481.6  298.19  5642.2  300.88  5853.2  306.26  5926.5  307.84
#Mann= 12 ,-1 , 0
  3453.7     .07       0  3994.9     .05       0  4805.5     .07       0
    4982     .05       0  5007.1     .07       0  5042.1     .05       0
  5252.4    .035       0  5285.3     .05       0  5436.8    .035       0
  5481.6     .05       0  5642.2     .07       0  5853.2     .05       0
Bank Sta=4982,5007.1
XS Rating Curve= 0 ,0
Exp/Cntr=0.3,0.1

Type RM Length L Ch R = 1 ,45274   ,557,557,557
BEGIN DESCRIPTION:
DENTON CREEK 2 46.0
END DESCRIPTION:
XS GIS Cut Line= 3
      2482575.01     13755024.97        2482975.       13753025.
        2483125.     13752225.02
#Sta/Elev= 30
  2965.6  313.28  3138.9  309.51  3398.4  306.33  3440.3  305.67  3756.2  301.82
  4117.9  296.61  4240.3  292.35  4291.3  293.46  4546.3   290.2  4668.6  287.12
  4852.2  286.72  4954.2  288.21  4964.4  287.79  4972.2  280.86  4972.7  280.36
  4997.4  280.86  5002.6  284.73  5007.7  284.73  5015.4  287.66  5066.6  287.58
    5084  286.67  5136.6  288.43  5273.3  287.71  5316.6  287.61    5402  289.75
  5414.7  291.59  5442.7  291.29  5493.5  295.18  5565.2  298.09  5819.1  307.01
#Mann= 10 ,-1 , 0
  2965.6     .07       0  3398.4     .05       0  3440.3     .07       0
  3756.2     .05       0  4972.2     .05       0  4997.4     .05       0
  5066.6      .1       0  5273.3     .05       0  5316.6     .07       0
  5565.2     .05       0
Bank Sta=4972.2,4997.4
XS Rating Curve= 0 ,0
Exp/Cntr=0.3,0.1

Type RM Length L Ch R = 1 ,44717   ,552,552,552
BEGIN DESCRIPTION:
DENTON CREEK 2 45.0
END DESCRIPTION:
XS GIS Cut Line= 3
      2482775.02     13754624.96        2483475.       13753075.
      2483674.99     13751475.04
#Sta/Elev= 30
    3299  306.71  3509.2  304.22  3957.3     303  4750.9  287.41  4864.3  285.23
  4990.9  287.22  5007.2  282.67  5007.7  282.17  5032.5  282.67  5037.5  287.66
  5148.5  287.26  5413.3  290.76  5512.1  292.61    5611  294.48  5826.1  299.53
  5848.7   301.4  5866.4  307.43  5906.7  302.85  5924.3  303.85  5929.4  301.62
  5967.2   308.4  6033.4  309.52  6324.6  326.48  6400.5  330.38  6420.7  334.62
  6430.7  335.02    6461  330.88  6501.3  334.74    6608  339.76  6612.1  339.86
#Mann= 11 ,-1 , 0
    3299     .05       0  4750.9      .1       0  5007.2     .05       0
  5032.5      .1       0  5148.5     .05       0  5413.3     .07       0
  5512.1    .035       0    5611     .07       0  6033.4     .05       0
  6324.6     .07       0    6608     .05       0
Bank Sta=5007.2,5032.5
XS Rating Curve= 0 ,0
Exp/Cntr=0.3,0.1

Type RM Length L Ch R = 1 ,44165   ,544,544,544
BEGIN DESCRIPTION:
DENTON CREEK 2 44.0
END DESCRIPTION:
XS GIS Cut Line= 3
      2483175.01     13754724.99        2483875.       13753325.
        2483775.     13751724.96
#Sta/Elev= 30
  3444.6  306.03    3534  304.16  4099.1  301.06  4207.7  301.25  4428.5  299.99
  4531.9  296.09    4571  296.43  4660.4  293.57  4688.4  291.55  4777.4  290.02
  4858.8  288.02  4942.8  286.75  4970.4  281.37  4974.8  280.96  4975.3  280.46
  5000.2  280.96  5001.4  285.41    5007  286.47  5059.9   284.7  5281.6  285.73
  5656.5  289.24  5761.6  290.59  5961.7  293.39  6011.8  294.92  6054.4  299.55
  6100.4  300.53  6130.1  302.31  6326.1  313.31  6502.7  324.16    6613  329.36
#Mann= 14 ,-1 , 0
  3444.6     .05       0  4099.1    .035       0  4207.7     .05       0
  4777.4    .035       0  4858.8     .05       0  4970.4      .1       0
  4974.8     .05       0  5000.2      .1       0  5281.6     .05       0
  5656.5    .035       0  5761.6     .07       0  6100.4     .05       0
  6130.1     .07       0  6326.1     .05       0
Bank Sta=4974.8,5000.2
XS Rating Curve= 0 ,0
Exp/Cntr=0.3,0.1

Type RM Length L Ch R = 1 ,43621   ,545,545,545
BEGIN DESCRIPTION:
DENTON CREEK 2 43.0
END DESCRIPTION:
XS GIS Cut Line= 3
      2484075.01     13754724.97        2484325.       13753325.
      2483924.99     13751724.96
#Sta/Elev= 30
  3582.6  303.22  4029.5  298.16  4151.4  293.46  4177.1  290.31  4183.4  291.49
  4212.4  289.41  4232.2  291.91  4237.3  289.14  4242.8   292.5  4273.3  295.57
  4455.3  293.43  4496.8  292.49  4521.7  289.15  4554.8  288.06  4654.3  284.88
    4801   283.3  4964.1  285.45  4977.8  283.73  4981.8  277.32  4982.3  276.82
  5007.3  277.32    5015  285.17  5099.2  286.39  5468.6  287.22  5635.3  289.64
  5768.9  289.93  5976.2  294.33  6399.9  313.06  6561.2   324.2    6654  327.93
#Mann= 11 ,-1 , 0
  3582.6     .05       0  4177.1     .07       0  4455.3    .035       0
  4554.8     .07       0  4654.3     .12       0  4981.8     .05       0
  5007.3     .12       0  5099.2     .05       0  5635.3    .035       0
  5768.9     .07       0  6399.9     .05       0
Bank Sta=4981.8,5007.3
XS Rating Curve= 0 ,0
Exp/Cntr=0.3,0.1

Type RM Length L Ch R = 1 ,43076   ,552,552,552
BEGIN DESCRIPTION:
DENTON CREEK 2 42.0
END DESCRIPTION:
XS GIS Cut Line= 3
      2484224.99     13754675.02        2484775.       13753575.
        2485125.     13752125.01
#Sta/Elev= 30
  3770.2   303.7  4239.8  297.55  4553.9  291.71  4575.2  291.24  4583.6  289.71
  4662.4  288.06  4718.1  286.48  4770.9  285.44  4829.6  282.59  4874.3  283.95
  4879.4  283.33  4951.5  283.24  4977.7  283.81  4984.5  276.38    4985  275.88
  5010.1  276.38  5018.4  282.79  5030.9  285.32  5089.4  284.29  5191.1  282.27
  5274.9  285.78  5411.6  283.78  5578.4  285.39  5648.2  284.29  5761.3   285.1
  5871.5  286.92  5936.2  286.82  6162.5  294.68  6389.6  305.33  6491.7  307.93
#Mann= 10 ,-1 , 0
  3770.2     .05       0  4553.9    .035       0  4662.4     .05       0
  4718.1    .035       0  4770.9     .05       0  4879.4     .12       0
  4951.5      .1       0  4984.5     .05       0  5010.1      .1       0
  5089.4     .05       0
Bank Sta=4984.5,5010.1
XS Rating Curve= 0 ,0
Exp/Cntr=0.3,0.1

Type RM Length L Ch R = 1 ,42524   ,507,507,507
BEGIN DESCRIPTION:
DENTON CREEK 2 41.0
END DESCRIPTION:
XS GIS Cut Line= 3
      2484324.98     13754825.04        2485175.       13753425.
        2485225.     13752274.96
#Sta/Elev= 30
  3357.5  307.06  3640.5  300.14  4231.1  290.61  4274.3  290.35  4305.1  289.23
  4326.7  286.89  4344.3  286.81  4519.6  283.79  4580.6  282.18  4749.2  283.08
  4819.9  282.29  4886.8  283.74  5005.4  282.95  5019.9   276.9  5022.6  276.13
  5023.1  275.63  5048.2  276.13  5055.4  281.73  5065.4  283.49  5118.3  283.57
  5205.6  281.27  5215.6  282.36  5355.7  284.57  5455.8  283.65  5555.9  284.24
  5736.1  287.15  5856.2  291.98  5966.3  297.66  6036.4  305.43  6146.5  309.68
#Mann= 8 ,-1 , 0
  3357.5     .05       0  4231.1    .035       0  4344.3     .05       0
  4519.6     .12       0  5019.9      .1       0  5022.6     .05       0
  5048.2      .1       0  5118.3     .05       0
Bank Sta=5022.6,5048.2
XS Rating Curve= 0 ,0
Exp/Cntr=0.3,0.1

Type RM Length L Ch R = 1 ,42017   ,2114,2114,2114
BEGIN DESCRIPTION:
DENTON CREEK 2 40.0
END DESCRIPTION:
XS GIS Cut Line= 3
      2484274.99     13755075.01        2485575.       13753525.
      2485324.99     13752374.97
#Sta/Elev= 30
  2990.8  312.44  3515.8  299.93  3651.9  299.62  3679.7  300.64  3714.8  296.02
  3729.6  295.97  3764.2  295.34  3786.3  298.69    3800  298.63  3821.5  296.42
  3899.5  294.92  4154.1  293.13  4279.6  290.53  4439.4   286.1  4758.2  284.67
  4892.8  282.01  4935.5  281.34  4942.9  276.01  4993.8  275.88  4994.3  275.38
  5019.5  275.88    5024  279.57  5038.4   283.1  5185.8  282.66  5453.9   280.9
  5607.4  284.72  5719.9  283.15  5832.5   284.7  5935.9  288.65  6190.7  308.34
#Mann= 9 ,-1 , 0
  2990.8     .05       0  3651.9     .07       0  3729.6     .05       0
  4154.1    .035       0  4279.6     .05       0  4892.8     .12       0
  4993.8     .05       0  5019.5     .12       0  5185.8     .05       0
Bank Sta=4993.8,5019.5
XS Rating Curve= 0 ,0
Exp/Cntr=0.3,0.1

Type RM Length L Ch R = 1 ,39903   ,544,544,544
BEGIN DESCRIPTION:
DENTON CREEK 2 39.0
END DESCRIPTION:
XS GIS Cut Line= 3
      2485225.01     13754624.99        2486825.       13752425.
        2486925.     13751675.02
#Sta/Elev= 30
  2280.1  298.22  2544.8  296.87  2680.8   294.6  2795.9  291.47  2960.2  288.98
  3088.8  289.56  3440.5  288.67  3662.3  286.66  3739.5  285.12    3813  286.49
  4091.2   287.5  4212.5  284.15  4342.3  282.97  4406.9  280.84  4695.9  280.18
  4821.5   279.1  4936.3  280.28  4957.5  280.41  5002.9  278.68  5007.5  273.29
    5008  272.79  5033.6  273.29    5037  278.02    5071   278.6  5110.1  283.74
  5131.5  285.01  5266.5  286.89  5630.4  296.08    5756  299.57    5757  299.57
#Mann= 7 ,-1 , 0
  2280.1     .05       0  4695.9     .12       0  4936.3     .05       0
  5007.5     .05       0  5033.6     .05       0  5630.4     .07       0
    5756     .05       0
Bank Sta=5007.5,5033.6
XS Rating Curve= 0 ,0
Exp/Cntr=0.3,0.1

Type RM Length L Ch R = 1 ,39359   ,569,569,569
BEGIN DESCRIPTION:
DENTON CREEK 2 38.0
END DESCRIPTION:
XS GIS Cut Line= 3
        2486975.       13754575.        2487175.       13752775.
        2487375.       13751325.
#Sta/Elev= 30
  3188.8  300.07  3329.7  298.59  3621.4  289.12  3732.1  286.75  4225.1  282.37
  4325.8   279.8  4478.5  279.78  4758.4  280.58    4859  278.13  4929.4  279.48
  4949.6  278.38  4966.6  271.81  4967.1  271.31  4992.8  271.81  4997.4  273.29
  5020.1  271.94  5040.9  277.52  5098.7  279.18  5179.7   278.2  5251.6  279.69
  5282.5  281.42  5328.6  280.41  5405.6  282.11  5454.1  281.94  5807.4  286.72
    5991  292.06  6059.6  296.92  6223.3  305.77  6372.7  311.79  6463.6  314.32
#Mann= 7 ,-1 , 0
  3188.8     .05       0  4478.5      .1       0  4966.6     .05       0
  4992.8      .1       0  5098.7     .05       0  6059.6     .07       0
  6223.3     .05       0
Bank Sta=4966.6,4992.8
XS Rating Curve= 0 ,0
Exp/Cntr=0.3,0.1

Type RM Length L Ch R = 1 ,38790   ,588,588,588
BEGIN DESCRIPTION:
DENTON CREEK 2 37.0
END DESCRIPTION:
XS GIS Cut Line= 3
      2487025.01     13754524.98        2487575.       13752975.
        2487475.     13751525.01
#Sta/Elev= 30
  3350.9  300.22  3546.2  296.51  3828.4  287.13  4316.5  284.63  4409.6  278.89
  4445.7  279.15    4465  276.46  4511.9   275.7  4527.7  274.92    4533  277.39
  4558.6  274.12  4563.9  276.64  4571.1  274.39  4594.8  273.44  4613.6  277.71
  4656.5  280.14  4974.3  279.12  4992.5  271.14    4993  270.64  5018.7  271.14
  5025.6  277.62  5035.7  278.89  5227.4  281.32  5360.2   283.4  5555.8   281.1
  5868.8  284.64  6068.1  288.92  6198.8  296.93  6389.6  308.81    6449  310.77
#Mann= 9 ,-1 , 0
  3350.9     .05       0  4511.9      .1       0  4992.5     .05       0
  5018.7      .1       0  5227.4     .05       0  5555.8     .07       0
  5868.8     .05       0  6198.8     .07       0  6389.6     .05       0
Bank Sta=4992.5,5018.7
XS Rating Curve= 0 ,0
Exp/Cntr=0.3,0.1

Type RM Length L Ch R = 1 ,38202   ,1625,1625,1625
BEGIN DESCRIPTION:
DENTON CREEK 2 36.0
END DESCRIPTION:
XS GIS Cut Line= 3
      2487124.99     13754425.01        2488125.       13752875.
      2487574.98     13751574.96
#Sta/Elev= 30
  3155.3  296.75  3235.5  295.35    3429  288.62  3690.8  285.41    4067   283.5
  4190.7  282.09  4275.6  279.86  4514.5  279.49  4680.8  276.53  4849.9  276.64
  4919.7  276.42  4992.3  278.09  4995.5  270.79    4996  270.29  5022.5  270.79
  5032.5  276.99  5038.2   277.5    5125  279.84  5191.2  281.78  5291.3  282.73
  5412.3  281.69  5480.5  281.15  5520.5  280.95  5628.7  281.74  5769.7  283.61
  5990.7   287.7    6158  296.16  6190.9   297.8    6386  308.55  6411.5  309.42
#Mann= 13 ,-1 , 0
  3155.3     .05       0  4849.9      .1       0  4995.5     .05       0
  5022.5      .1       0    5125     .05       0  5412.3    .035       0
  5480.5     .05       0  5520.5    .035       0  5628.7     .05       0
  5769.7    .035       0    6158     .05       0  6190.9    .035       0
    6386     .05       0
Bank Sta=4995.5,5022.5
XS Rating Curve= 0 ,0
Exp/Cntr=0.3,0.1

Type RM Length L Ch R = 1 ,36577   ,567,567,567
BEGIN DESCRIPTION:
DENTON CREEK 2 35.0
END DESCRIPTION:
XS GIS Cut Line= 3
      2490175.03     13753775.03        2489425.       13753175.
      2487824.97     13751574.97
#Sta/Elev= 30
  4044.9  293.73  4181.6  288.06  4229.8  286.74  4304.9  282.37  4429.1   279.1
  4479.6  280.85  4621.2  279.63  4713.3   280.4  4863.7  276.18  4913.4  272.72
  4934.2  272.85  4947.8  274.77  4977.4  275.88  4981.2  267.69  4981.9  267.19
  5015.2  267.69  5019.6  275.19  5033.7  276.16  5076.1  273.67  5104.4  275.29
  5161.4  274.85  5302.4  276.82  5394.3  275.43    5557  280.93  5797.4  279.77
  6009.5  282.45  6108.5  281.06  6292.3  281.88  6667.1  289.11  7268.2  303.33
#Mann= 7 ,-1 , 0
  4044.9     .05       0  4181.6    .035       0  4304.9     .05       0
  4947.8      .1       0  4981.2     .05       0  5015.2      .1       0
  5161.4     .05       0
Bank Sta=4981.2,5015.2
XS Rating Curve= 0 ,0
Exp/Cntr=0.3,0.1

Type RM Length L Ch R = 1 ,36010   ,564,564,564
BEGIN DESCRIPTION:
DENTON CREEK 2 34.0
END DESCRIPTION:
XS GIS Cut Line= 3
      2490324.98     13753224.98        2489775.       13752775.
        2489225.       13751175.
#Sta/Elev= 30
  4282.9  292.59  4339.4  291.91  4389.1  291.02  4562.1  282.88  4617.4  279.07
  4714.7  277.35  4721.7  277.04  4851.4  275.92    4916  273.93  4986.3  274.17
  4990.3  271.21  4996.2  271.21  4997.6  267.35  4998.2  266.85  5031.8  267.35
  5035.1  273.23  5040.4  274.48  5109.9   273.9  5191.3  274.32  5215.6  273.23
  5259.1  274.36    5279  273.12    5285  275.12  5296.6  275.61    5330   275.2
  5479.9  277.18  5723.1   276.1  6050.2  279.11  6487.6  289.79  6685.4  296.19
#Mann= 10 ,-1 , 0
  4282.9     .05       0  4339.4     .07       0  4562.1    .035       0
  4714.7     .05       0  4721.7      .1       0  4997.6     .05       0
  5031.8      .1       0  5109.9     .05       0  5296.6     .12       0
    5330     .05       0
Bank Sta=4997.6,5031.8
XS Rating Curve= 0 ,0
Exp/Cntr=0.3,0.1

Type RM Length L Ch R = 1 ,35446   ,522,522,522
BEGIN DESCRIPTION:
DENTON CREEK 2 33.0
END DESCRIPTION:
XS GIS Cut Line= 3
      2490424.99     13753274.98        2490075.       13752325.
      2489225.01     13751025.02
#Sta/Elev= 30
  3982.1     295  4019.6  294.11  4109.9  292.17  4115.1  292.02  4169.3  291.06
  4216.7  288.66  4322.7  283.98  4525.6  279.23  4725.8   276.1  4909.2  273.73
  4941.2  271.16  4962.5  274.04  4984.6  274.74  4990.7  267.13  4991.4  266.63
  5025.4  267.13  5038.3  274.47  5044.2  275.32  5066.2  273.81  5119.4  273.25
  5161.8  273.61  5173.9  274.85    5189  273.99  5204.1  275.07  5225.2  274.74
  5261.4  276.28  5327.8  275.41    5572  276.07  6425.6  297.58  6547.7  299.78
#Mann= 10 ,-1 , 0
  3982.1     .05       0  4019.6     .07       0  4109.9     .05       0
  4115.1     .07       0  4216.7    .035       0  4322.7     .05       0
  4725.8      .1       0  4990.7     .05       0  5025.4      .1       0
  5119.4     .05       0
Bank Sta=4990.7,5025.4
XS Rating Curve= 0 ,0
Exp/Cntr=0.3,0.1

Type RM Length L Ch R = 1 ,34924   ,518,518,518
BEGIN DESCRIPTION:
DENTON CREEK 2 32.0
END DESCRIPTION:
XS GIS Cut Line= 3
      2491524.97     13752524.98        2490275.       13751875.
      2489475.02     13751075.02
#Sta/Elev= 30
  3590.9  299.55  3671.1  298.04  3776.6  293.99  3820.2  290.16  3850.1  285.34
  3886.5  283.52  4146.2   278.4  4273.2  277.07  4323.5  277.97  4413.7  277.52
  4538.5  274.44  4655.8  274.81  4740.5  274.44  4830.7  272.21  4864.5  274.12
  4941.7  275.18  4963.8  274.24  4968.4  267.22  4969.2  266.72  5003.3  267.22
  5013.9  273.96  5042.2  273.64  5070.5  269.63  5084.6  273.81  5087.6  273.75
  5183.6  272.41  5282.6   277.2  5367.5     279    5721  282.21  6131.1  293.98
#Mann= 6 ,-1 , 0
  3590.9     .07       0  3776.6     .05       0  4655.8      .1       0
  4968.4     .05       0  5003.3      .1       0  5087.6     .05       0
Bank Sta=4968.4,5003.3
XS Rating Curve= 0 ,0
Exp/Cntr=0.3,0.1

Type RM Length L Ch R = 1 ,34406   ,567,567,567
BEGIN DESCRIPTION:
DENTON CREEK 2 31.0
END DESCRIPTION:
XS GIS Cut Line= 3
      2492175.04     13752975.03        2490625.       13751575.
      2489925.01     13750775.02
#Sta/Elev= 30
  2906.4  321.08  2913.5  319.29  3158.5  310.97  3189.7  309.62  3361.8  306.97
  3624.5  300.21  3784.1  294.34    3904  285.27  3933.8  283.39  4032.1  280.21
  4495.4  275.71  4704.8  272.58  4751.9  273.66  4825.1  271.47  4959.6  274.22
  4967.1   273.2  4974.2  265.92    4975  265.42  5009.2  265.92  5016.5  272.54
  5023.1  273.32  5135.6  273.72  5241.2  274.42  5291.3  275.71  5382.3  276.24
  5436.1  276.93  5619.2   284.1  5836.3  287.95  6015.5  294.72  6058.1  295.84
#Mann= 19 ,-1 , 0
  2906.4     .07       0  3158.5    .035       0  3189.7     .07       0
  3361.8    .035       0  3624.5     .07       0    3904     .05       0
  3933.8     .07       0  4032.1     .05       0  4495.4     .12       0
  4751.9      .1       0  4974.2     .05       0  5009.2      .1       0
  5135.6     .12       0  5241.2      .1       0  5291.3     .07       0
  5382.3    .035       0  5436.1     .07       0  5836.3    .035       0
  6015.5     .05       0
Bank Sta=4974.2,5009.2
XS Rating Curve= 0 ,0
Exp/Cntr=0.3,0.1

Type RM Length L Ch R = 1 ,33839   ,574,574,574
BEGIN DESCRIPTION:
DENTON CREEK 2 30.0
END DESCRIPTION:
XS GIS Cut Line= 3
        2492225.     13752925.01        2491125.       13751375.
      2490125.03     13750225.03
#Sta/Elev= 30
  3099.4  322.82  3239.8  319.51    3363  312.26  3374.8   311.8  3486.2  307.87
  3558.3  306.68  3831.4  293.95  3977.7  289.14  4192.8  279.63  4225.3  278.84
  4348.5   276.7  4356.4  276.51  4471.7  275.75  4500.6  275.67  4666.2  274.03
  4835.2  271.56  4977.9  272.65  4979.5  266.32  4980.2  265.82  5014.5  266.32
  5021.4  271.65  5049.9  274.49    5255  271.66  5590.9  274.18  5921.6  279.32
  6091.4  286.53  6110.7  287.27  6317.4  302.48  6432.6  313.24    6524  319.16
#Mann= 20 ,-1 , 0
  3099.4     .07       0  3239.8    .035       0    3363     .05       0
  3374.8     .07       0  3486.2     .05       0  3977.7     .07       0
  4192.8     .05       0  4225.3     .07       0  4348.5     .05       0
  4356.4     .07       0  4471.7     .05       0  4500.6     .07       0
  4666.2      .1       0  4979.5     .05       0  5014.5      .1       0
  5590.9     .05       0  6091.4     .07       0  6110.7     .05       0
  6317.4     .07       0  6432.6     .05       0
Bank Sta=4979.5,5014.5
XS Rating Curve= 0 ,0
Exp/Cntr=0.3,0.1

Type RM Length L Ch R = 1 ,33265   ,572,572,572
BEGIN DESCRIPTION:
DENTON CREEK 2 29.0
END DESCRIPTION:
XS GIS Cut Line= 3
      2492625.01     13752475.01        2491375.       13750925.
      2490625.02     13750125.02
#Sta/Elev= 30
  3008.1  317.86  3064.9  315.25  3122.5  317.24  3192.8  311.92  3413.6  306.45
    3450  303.62  3634.3  299.41  3722.9  290.17  3795.7  283.47    3855  279.05
  3984.6   276.9  4298.2  271.83  4373.2  269.13  4494.7  274.65  4686.7  272.43
  4921.8   274.4  4985.7  272.48  4992.2  270.17  4995.5  265.85  4996.3  265.35
    5031  265.85  5065.7  271.74  5147.3  275.58  5324.9  282.19  5424.6  282.09
  5664.4  276.83  5841.2  288.52  5926.2   298.7  6019.6  306.19  6095.9  308.41
#Mann= 12 ,-1 , 0
  3008.1     .07       0    3450     .05       0  3722.9     .07       0
  3795.7     .05       0  3984.6     .07       0  4298.2      .1       0
  4995.5     .05       0    5031      .1       0  5065.7     .12       0
  5147.3     .07       0  5424.6     .12       0  6019.6     .07       0
Bank Sta=4995.5,5031
XS Rating Curve= 0 ,0
Exp/Cntr=0.3,0.1

Type RM Length L Ch R = 1 ,32693   ,535,535,535
BEGIN DESCRIPTION:
DENTON CREEK 2 28.0
END DESCRIPTION:
XS GIS Cut Line= 3
        2492425.       13752125.        2491775.       13751025.
      2491224.98     13750024.97
#Sta/Elev= 30
  3722.2  310.32  3942.7  303.33  4012.8   290.8    4214  277.62  4270.5  276.16
  4441.7  273.21  4612.9  273.41  4623.7  273.23    4875  271.47  4890.7  266.07
  4896.5  269.91  4900.8  264.56  4901.6  264.06  4936.3  264.56  4992.1  266.25
  5007.9  270.88  5013.6  267.06  5029.7  271.07  5035.4  264.64  5051.5  271.27
  5057.2  265.64  5073.3   265.1  5095.1   266.2  5111.2  272.29  5116.9  267.35
    5133  272.83  5272.7   274.8  5800.1  281.42  6023.4  289.07  6141.2  290.64
#Mann= 11 ,-1 , 0
  3722.2     .07       0    4214     .05       0  4270.5     .07       0
  4441.7      .1       0  4612.9     .07       0  4623.7      .1       0
  4900.8     .05       0  4936.3      .1       0  5272.7     .05       0
  5800.1    .035       0  6023.4     .12       0
Bank Sta=4900.8,4936.3
XS Rating Curve= 0 ,0
Exp/Cntr=0.3,0.1

Type RM Length L Ch R = 1 ,32158   ,562,562,562
BEGIN DESCRIPTION:
DENTON CREEK 2 27.0
END DESCRIPTION:
XS GIS Cut Line= 3
      2492575.01     13751925.02        2492175.       13751125.
      2491175.02     13749525.04
#Sta/Elev= 30
  4109.9  315.89    4163   314.9    4191  312.96  4221.7  299.16  4258.1   293.8
  4333.5  289.74  4453.7  280.77  4516.3  279.07  4654.8  274.84  4724.6  273.58
  4766.5  273.69    4859  274.39  4951.2  272.19  4955.8  264.69  4956.6  264.19
  4991.4  264.69  5001.6   270.8    5012  272.02  5200.7  270.33  5358.7  272.61
  5410.6   271.9  5461.6  273.56  5560.9  274.66  5830.4  275.43  5944.4  278.51
  6086.3  282.37  6170.7  282.95    6354  286.07  6690.8  288.22  6891.1  293.86
#Mann= 13 ,-1 , 0
  4109.9     .07       0  4516.3     .05       0  4654.8     .12       0
  4724.6     .05       0  4766.5     .12       0    4859      .1       0
  4955.8     .05       0  4991.4      .1       0  5461.6     .07       0
  5560.9     .05       0  5944.4    .035       0  6170.7     .07       0
  6690.8     .12       0
Bank Sta=4955.8,4991.4
XS Rating Curve= 0 ,0
Exp/Cntr=0.3,0.1

Type RM Length L Ch R = 1 ,31596   ,553,553,553
BEGIN DESCRIPTION:
DENTON CREEK 2 26.0
END DESCRIPTION:
XS GIS Cut Line= 3
      2492974.98     13751074.99        2492625.       13750825.
        2491175.       13749375.
#Sta/Elev= 30
  4565.1  293.64  4588.2  292.52  4774.8  280.02  4845.3  277.24  4893.4  277.13
  4922.7  276.06    4946  271.92  4973.1   271.1  4974.3  264.47  4975.1  263.97
    5010  264.47  5023.5     271  5065.9   271.2  5122.5  269.31  5292.2  272.06
  5380.9  271.74  5420.6  271.72  5524.2   273.5  5603.3  272.81  5724.9  273.89
  5829.6  276.33  5956.9  277.48  6055.9  276.84  6140.7  277.85  6183.1  279.64
  6225.6  282.89  6579.1  284.88  6801.3  289.95  6960.9  295.81  7045.8  297.29
#Mann= 12 ,-1 , 0
  4565.1     .12       0  4588.2     .07       0  4774.8     .12       0
  4893.4      .1       0  4974.3     .05       0    5010      .1       0
  5380.9     .07       0  5420.6     .12       0  5524.2     .07       0
  5724.9     .05       0  5956.9     .07       0  6801.3     .12       0
Bank Sta=4974.3,5010
XS Rating Curve= 0 ,0
Exp/Cntr=0.3,0.1

Type RM Length L Ch R = 1 ,31043   ,584,584,584
BEGIN DESCRIPTION:
DENTON CREEK 2 25.0
END DESCRIPTION:
XS GIS Cut Line= 3
      2493075.01     13751075.01        2492775.       13750325.
        2491625.       13748725.
#Sta/Elev= 30
  4186.6  296.68    4246  294.02  4380.5  286.73  4461.6  279.89    4573  274.43
    4691   272.5  4769.6  271.08  4811.3  271.96  4979.6  270.97  5001.8  270.08
  5007.9  265.21  5013.3  264.22  5014.1  263.72  5049.1  264.22  5052.1  269.53
  5066.8  271.96  5241.3  272.26  5302.3  271.96  5408.1  273.47  5638.9   275.1
  6012.1  280.04  6118.9  279.57  6305.5  282.82  6312.1  283.74  6320.3  283.02
  6398.3  286.02  6427.1  285.74  6584.2  290.23    6861  300.12  6964.8  303.71
#Mann= 9 ,-1 , 0
  4186.6     .07       0    4246     .12       0  4461.6     .07       0
    4691      .1       0  5013.3     .05       0  5049.1      .1       0
  5241.3     .12       0  5408.1     .07       0    6861    .035       0
Bank Sta=5013.3,5049.1
XS Rating Curve= 0 ,0
Exp/Cntr=0.3,0.1

Type RM Length L Ch R = 1 ,30459   ,549,549,549
BEGIN DESCRIPTION:
DENTON CREEK 2 24.0
END DESCRIPTION:
XS GIS Cut Line= 3
        2493375.     13751475.03        2493175.       13749925.
      2491574.97     13748474.97
#Sta/Elev= 30
  3432.4  314.43  3623.4  297.49    3745   294.6  4080.3  279.33  4118.2  277.35
  4264.4  273.19    4602  271.95  4783.5  268.82  4944.9  271.97  4953.1  271.74
    4965   265.4  4984.5  264.47  4985.3  263.97  5020.3  264.47  5030.8  270.79
  5099.5  269.92  5349.1  276.27  5508.5  277.85  5659.8  276.19  5717.6  276.91
  5792.5  278.31  6085.1  283.34  6375.7  285.29  6744.6  295.96  6793.3  297.45
    6815  300.39  6821.7   298.9  6850.1  299.59    7007  305.28  7154.6  310.13
#Mann= 14 ,-1 , 0
  3432.4     .07       0  4080.3     .12       0  4118.2     .07       0
  4264.4      .1       0  4984.5     .05       0  5020.3      .1       0
  5099.5     .12       0  5508.5     .05       0  5659.8     .07       0
  5717.6     .05       0  5792.5     .07       0  6085.1     .05       0
  6744.6    .035       0    7007     .05       0
Bank Sta=4984.5,5020.3
XS Rating Curve= 0 ,0
Exp/Cntr=0.3,0.1

Type RM Length L Ch R = 1 ,29910   ,1652,1652,1652
BEGIN DESCRIPTION:
DENTON CREEK 2 23.0
END DESCRIPTION:
XS GIS Cut Line= 3
      2494074.99     13751224.98        2493575.       13749675.
      2492425.02     13748075.03
#Sta/Elev= 30
  3376.7  306.02    3585  288.51    3934  271.97  3961.3  271.59  4038.3   268.3
  4140.3  271.32  4390.7  269.96  4485.8  269.73  4690.1  270.87  4791.8  267.04
  4931.8   270.8  4971.3  264.37  4972.1  263.87  5007.4  264.37  5008.4   270.3
  5042.1  272.16  5206.5  271.26  5593.4   272.9  5629.1  276.95  5643.7  277.51
  5664.6  270.93  5685.5  269.72  5765.3  269.64  5825.7  276.06  5982.8  278.05
  6066.4  277.57  6366.6   279.3  6646.9  286.09  6919.4  291.85  6975.7  292.54
#Mann= 16 ,-1 , 0
  3376.7     .05       0    3934     .07       0  3961.3     .05       0
  4038.3     .12       0  4390.7     .07       0  4485.8      .1       0
  4971.3     .05       0  5007.4      .1       0  5206.5     .05       0
  5629.1     .07       0  5825.7     .05       0  5982.8    .035       0
  6066.4     .05       0  6366.6     .07       0  6646.9     .05       0
  6919.4    .035       0
Bank Sta=4971.3,5007.4
XS Rating Curve= 0 ,0
Exp/Cntr=0.3,0.1

Type RM Length L Ch R = 1 ,28258   ,1221,1221,1221
BEGIN DESCRIPTION:
DENTON CREEK 2 22.0
END DESCRIPTION:
XS GIS Cut Line= 3
        2494425.       13751025.        2494625.       13750675.
      2492325.01     13747475.02
#Sta/Elev= 30
  4587.1  289.81  4805.9   283.3    4852  279.58  4904.5  269.69  4944.8  266.96
  4987.3  264.06  5056.9  265.81  5065.4  262.87  5066.3  262.37  5101.6  262.87
  5162.6  268.61  5225.9  263.44  5255.6  266.11  5461.8  268.43  5516.3  268.81
  5706.1  271.65  6200.6  269.89  6919.8  272.04  7004.6  272.77  7341.2  275.02
  7376.8  278.28  7397.7  275.84  7484.3  279.93  7863.3  282.21  8354.3  290.79
  8463.7  292.73  8615.3  294.32  8776.1  296.99  8789.9  297.19    8931  299.33
#Mann= 20 ,-1 , 0
  4587.1     .05       0  4904.5     .12       0  4944.8      .1       0
  5056.9     .12       0  5065.4     .05       0  5101.6      .1       0
  5255.6     .12       0  5461.8     .07       0  5516.3     .12       0
  5706.1      .1       0  6200.6     .05       0  6919.8     .07       0
  7004.6     .05       0  7484.3     .07       0  7863.3     .05       0
  8354.3     .07       0  8463.7     .05       0  8615.3     .07       0
  8776.1    .035       0  8789.9     .07       0
Bank Sta=5065.4,5101.6
XS Rating Curve= 0 ,0
Exp/Cntr=0.3,0.1
