--- EAST TINSLEY CREEK.prj (project) ---

Proj Title=EAST TINSLEY CREEK Base Level Engineering
Current Plan=p01
Default Exp/Contr=0.3,0.1
English Units
Geom File=g01
Flow File=f01
Plan File=p01
Y Axis Title=Elevation
X Axis Title(PF)=Main Channel Distance
X Axis Title(XS)=Station
BEGIN DESCRIPTION:
EAST TINSLEY CREEK
END DESCRIPTION:
DSS Export Rating Curves= 0
DSS Export Rating Curve Sorted= 0
DSS Export Volume Flow Curves= 0
DXF OffsetX= 0
DXF OffsetY= 0
DXF ScaleX= 1
DXF ScaleY= 10

--- EAST TINSLEY CREEK.p01 (plan) ---

Plan Title=Multiple Run
Short Identifier=Multiple
Geom File=g01
Flow File=f01
Subcritical Flow
K Sum by GR= 0
Std Step Tol= 0.01
Critical Tol= 0.01
Num of Std Step Trials= 20
Max Error Tol= 0.3
Flow Tol Ratio= 0.001
Split Flow NTrial= 30
Split Flow Tol= 0.02
Split Flow Ratio= 0.02
Log Output Level= 0
Friction Slope Method= 1
Unsteady Friction Slope Method= 2
Unsteady Bridges Friction Slope Method= 1
Parabolic Critical Depth
Global Vel Dist=  1 , 1 , 1
Global Log Level= 0
CheckData=True
Encroach Param= -1, 0, 0, 0
BEGIN DESCRIPTION:
Multiple Run
END DESCRIPTION:

--- EAST TINSLEY CREEK.f01 (steady flow) ---

Flow Title=Multiple
Number of Profiles=7
Profile Names=10-year,25-year,50-year,1pct_min,100-year,1pct_plu,500-year
River Rch & RM= EAST TINSLEY CRE,Reach-1,33134
     818    1333    1805    1183    2360    4708    3995
River Rch & RM= EAST TINSLEY CRE,Reach-1,27407
    1053    1727    2345    1539    3071    6127    5218
River Rch & RM= EAST TINSLEY CRE,Reach-1,20991
    1296    2146    2932    1935    3860    7702    6631
River Rch & RM= EAST TINSLEY CRE,Reach-1,19241
    1496    2488    3408    2253    4496    8970    7754
River Rch & RM= EAST TINSLEY CRE,Reach-1,15228
    1635    2720    3727    2463    4915    9807    8472
River Rch & RM= EAST TINSLEY CRE,Reach-1,9842
    1753    2913    3988    2632    5252   10478    9028
River Rch & RM= EAST TINSLEY CRE,Reach-1,1738
    1813    3018    4137    2733    5453   10880    9392
Boundary for River Rch & Prof#=EAST TINSLEY CRE,Reach-1,1
Up Type=0
Dn Type=3
Dn Slope=0.005
Boundary for River Rch & Prof#=EAST TINSLEY CRE,Reach-1,2
Up Type=0
Dn Type=3
Dn Slope=0.005
Boundary for River Rch & Prof#=EAST TINSLEY CRE,Reach-1,3
Up Type=0
Dn Type=3
Dn Slope=0.005
Boundary for River Rch & Prof#=EAST TINSLEY CRE,Reach-1,4
Up Type=0
Dn Type=3
Dn Slope=0.005
Boundary for River Rch & Prof#=EAST TINSLEY CRE,Reach-1,5
Up Type=0
Dn Type=3
Dn Slope=0.005
Boundary for River Rch & Prof#=EAST TINSLEY CRE,Reach-1,6
Up Type=0
Dn Type=3
Dn Slope=0.005
Boundary for River Rch & Prof#=EAST TINSLEY CRE,Reach-1,7
Up Type=0
Dn Type=3
Dn Slope=0.005

--- EAST TINSLEY CREEK.g01 (geometry) ---

Geom Title=Existing Conditions
Program Version=4.10

River Reach=EAST TINSLEY CRE,Reach-1
Reach XY= 30
        2481375.       13775125.      2482480.18     13773780.41
      2483064.68     13773485.19      2483572.86     13772519.03
      2483430.46     13772122.55      2483969.42     13771870.24
      2484174.06     13771414.51      2483725.46     13770914.48
      2483871.84     13769783.34      2482876.04     13768314.56
      2482967.79     13766974.65      2482732.21     13766875.35
      2483082.47     13765721.38      2485365.87     13764181.74
       2485567.7     13762924.92      2485225.94     13762364.51
      2485378.45     13761676.19      2485958.72     13761591.75
      2485724.41       13761000.      2485979.95     13760422.49
      2487019.54     13759727.45      2487175.32     13758749.89
       2486978.1     13758476.65      2487617.17     13758228.22
      2487432.69     13757568.53      2488671.55     13757023.52
      2488025.03     13756290.42      2488471.55     13755773.75
      2488483.28     13754721.78        2489175.       13753325.

Type RM Length L Ch R = 1 ,33134   ,299,299,299
BEGIN DESCRIPTION:
X19090
END DESCRIPTION:
XS GIS Cut Line= 3
      2481750.64     13775206.07      2481372.99     13775090.26
      2480824.19     13775024.81
#Sta/Elev= 30
    4607  375.97  4622.9  375.36  4686.1  375.15    4707  373.67  4790.7  372.39
  4802.3  371.54  4811.6  372.04  4822.1  371.97  4867.8  370.48  4895.3  370.02
  4933.3  368.48  4938.5  367.76  4958.1  367.24  4989.4  364.66  5002.6  364.45
  5002.9  363.95  5006.4  363.95  5006.6  364.45  5130.9  366.16  5161.1  367.38
  5181.3  369.13    5282  371.85  5332.3  372.25  5352.5  373.06  5392.7  373.45
  5402.8  373.94  5412.9  373.66  5483.4  374.11  5533.7  374.91  5554.7  374.81
#Mann= 3 ,-1 , 0
    4607     .05       0  5002.6     .05       0  5006.6     .05       0
Bank Sta=5002.6,5006.6
XS Rating Curve= 0 ,0
Exp/Cntr=0.3,0.1

Type RM Length L Ch R = 1 ,32835   ,470,470,470
BEGIN DESCRIPTION:
EAST TINSLEY CREEK 65.0
END DESCRIPTION:
XS GIS Cut Line= 3
      2481674.98     13775074.98        2481475.       13774825.
      2481224.98       13774775.
#Sta/Elev= 30
    4685  373.14  4706.6  373.25    4721   372.4  4756.2  371.11  4762.6  370.26
    4785  369.88  4791.4  370.27  4799.4   369.3  4820.2  369.03  4849.1  367.82
  4877.1  367.13  4933.9  363.81  4954.7  363.17  4962.7  363.28  4983.5  362.86
  4989.5  362.52  4989.8  362.02  4993.3  362.02  4993.5  362.52  4997.9  363.04
  5007.7  362.85  5025.5  363.44  5035.7  364.17  5056.1     365  5086.7  367.56
  5096.9  367.97  5178.5  370.26  5198.9  371.12  5219.3  371.13  5260.1   371.9
#Mann= 3 ,-1 , 0
    4685     .05       0  4989.5     .05       0  4993.5     .05       0
Bank Sta=4989.5,4993.5
XS Rating Curve= 0 ,0
Exp/Cntr=0.3,0.1

Type RM Length L Ch R = 1 ,32365   ,447,447,447
BEGIN DESCRIPTION:
EAST TINSLEY CREEK 64.0
END DESCRIPTION:
XS GIS Cut Line= 3
      2481974.99     13774824.98        2481825.       13774525.
        2481675.       13774225.
#Sta/Elev= 30
  4669.2  373.61  4705.5  372.24  4713.9  372.35  4722.3   371.7  4727.9  371.86
  4733.6  371.24    4781  368.55    4795  368.45  4834.1  366.13  4848.1   366.5
  4878.8  364.89  4901.2  361.81  4994.2  360.09  4994.5  359.59    4998  359.59
  4998.2  360.09  5001.8  360.89  5026.9  361.73  5035.3  361.31  5040.9  362.01
  5071.7  363.21  5080.1  363.76    5094   365.6  5116.4  366.58  5197.4  367.51
  5205.8  368.38  5219.8  367.77  5272.9  369.05  5281.3   368.8    5340  370.53
#Mann= 4 ,-1 , 0
  4669.2     .12       0  4733.6     .07       0  4994.2     .05       0
  4998.2     .07       0
Bank Sta=4994.2,4998.2
XS Rating Curve= 0 ,0
Exp/Cntr=0.3,0.1

Type RM Length L Ch R = 1 ,31918   ,442,442,442
BEGIN DESCRIPTION:
EAST TINSLEY CREEK 63.0
END DESCRIPTION:
XS GIS Cut Line= 3
      2482275.04     13774425.03        2482125.       13774325.
      2481875.03     13774025.03
#Sta/Elev= 30
  4805.5  368.13  4834.1  367.35  4877.7  364.67  4885.2  364.79  4906.2  363.74
  4949.8  364.38  4963.3  361.03  4972.3  360.43  4978.3  358.95  4982.8  358.39
    4993  357.96  5007.3  359.02  5028.1  358.47  5040.5  357.24  5040.7  356.74
  5044.2  356.74  5044.5  357.24  5050.3  358.72  5056.8  358.81  5063.9  359.96
  5085.4  361.17    5114  361.75  5128.4  361.47  5198.7   364.2  5298.2  366.31
    5334  367.96  5348.4  368.11  5362.7  368.92  5369.2  369.88  5376.3  369.95
#Mann= 3 ,-1 , 0
  4805.5     .07       0  5040.5     .05       0  5044.5     .07       0
Bank Sta=5040.5,5044.5
XS Rating Curve= 0 ,0
Exp/Cntr=0.3,0.1

Type RM Length L Ch R = 1 ,31476   ,443,443,443
BEGIN DESCRIPTION:
EAST TINSLEY CREEK 62.0
END DESCRIPTION:
XS GIS Cut Line= 3
        2482525.     13774324.99        2482325.       13774025.
      2482174.99     13773874.99
#Sta/Elev= 30
  4634.4  373.14  4641.9  372.57  4662.9  371.84    4678   370.5    4720  368.51
  4756.1  367.53  4771.1   366.6  4792.1  366.14  4858.2  362.95  4879.3  363.43
  4915.3  361.41  4922.8  360.72  4936.4  358.58  4958.9  357.57  4972.4     358
  4981.4  357.68  4998.5  357.97  5009.1   356.6  5021.2  355.81  5021.5  355.31
    5025  355.31  5025.2  355.81  5037.4  357.88  5051.5  359.71  5065.7  360.35
  5093.9  362.59  5122.2  363.22  5150.5  365.73  5171.7  366.29  5207.1  367.88
#Mann= 3 ,-1 , 0
  4634.4     .07       0  5021.2     .05       0  5025.2     .07       0
Bank Sta=5021.2,5025.2
XS Rating Curve= 0 ,0
Exp/Cntr=0.3,0.1

Type RM Length L Ch R = 1 ,31033   ,409,409,409
BEGIN DESCRIPTION:
EAST TINSLEY CREEK 61.0
END DESCRIPTION:
XS GIS Cut Line= 3
      2482674.99     13773974.97        2482575.       13773725.
      2482324.98     13773624.99
#Sta/Elev= 30
  4734.9  364.73  4756.4  363.89  4773.9  362.39  4779.3  362.91  4788.7  362.54
  4842.6  359.19    4852  359.44  4864.1  358.29  4905.8  356.36  4982.6  355.68
  4994.7  354.87  5001.4  353.18  5011.5  353.11  5011.8  352.61  5015.3  352.61
  5015.5  353.11  5018.9  354.06  5036.4  356.29  5079.5  358.25  5090.3  357.93
  5126.6  359.57  5133.4  361.21  5144.1  361.35  5175.1  364.13  5180.5  363.09
  5187.2  364.06  5210.1  364.56    5229  366.77  5258.6  368.56  5273.4  368.81
#Mann= 3 ,-1 , 0
  4734.9     .07       0  5011.5     .05       0  5015.5     .07       0
Bank Sta=5011.5,5015.5
XS Rating Curve= 0 ,0
Exp/Cntr=0.3,0.1

Type RM Length L Ch R = 1 ,30624   ,448,448,448
BEGIN DESCRIPTION:
EAST TINSLEY CREEK 60.0
END DESCRIPTION:
XS GIS Cut Line= 3
      2483025.01     13773825.01        2482825.       13773525.
      2482725.02     13773375.04
#Sta/Elev= 30
  4639.3  367.37  4646.8  366.93  4661.8  366.99  4675.4  365.86  4747.5  362.49
    4755  362.64    4761  361.97  4806.1  361.06  4812.1  359.79  4819.6  358.96
  4848.1  357.19  4899.2  354.98  4935.3  354.45  4941.3   354.9  4969.3  352.54
  4969.6  352.04  4973.1  352.04  4973.3  352.54  4977.3  353.43  4986.3  352.69
  5002.9  352.83  5007.4  353.46  5028.4  354.61  5043.4  356.28    5072  358.47
  5100.5  359.24  5115.5  361.16  5121.6  360.94  5144.1  362.75  5180.1  363.82
#Mann= 3 ,-1 , 0
  4639.3     .07       0  4969.3     .05       0  4973.3     .07       0
Bank Sta=4969.3,4973.3
XS Rating Curve= 0 ,0
Exp/Cntr=0.3,0.1

Type RM Length L Ch R = 1 ,30176   ,461,461,461
BEGIN DESCRIPTION:
EAST TINSLEY CREEK 59.0
END DESCRIPTION:
XS GIS Cut Line= 3
      2483275.04     13773425.02        2483075.       13773325.
      2482874.97     13773224.98
#Sta/Elev= 30
  4775.9  362.33  4784.3  361.88  4812.3   361.5  4820.7  359.73  4851.4   357.8
  4865.4  357.23  4873.8  357.39  4887.8  356.34  4910.1  355.72  4918.5  355.86
  4940.9  354.44  4968.8   353.9  4971.6  353.29  4985.6  351.76  5002.4  351.51
  5007.9  350.78  5013.5  351.18  5019.9  350.73  5020.2  350.23  5023.7  350.23
  5023.9  350.73  5030.3  351.53  5035.9  351.36  5052.7  352.43    5089  353.84
  5156.1  360.26  5186.8  361.63  5192.4  362.31  5200.8  362.14  5223.2  363.02
#Mann= 3 ,-1 , 0
  4775.9     .07       0  5019.9     .05       0  5023.9     .07       0
Bank Sta=5019.9,5023.9
XS Rating Curve= 0 ,0
Exp/Cntr=0.3,0.1

Type RM Length L Ch R = 1 ,29715   ,463,463,463
BEGIN DESCRIPTION:
EAST TINSLEY CREEK 58.0
END DESCRIPTION:
XS GIS Cut Line= 3
      2483524.98     13773224.98        2483325.       13772975.
      2483125.03     13772875.02
#Sta/Elev= 30
  4680.1  362.22  4730.5  361.47  4744.1  359.61  4765.7  358.93  4780.1  359.31
  4786.5   358.3  4850.6  355.98  4885.8  352.95  4893.8  351.62  4900.2  351.51
  4908.2   350.4  4914.6  350.53  4922.6   349.5    4929  350.45  4936.2  350.22
  4943.4  348.95  4957.8  349.52  4976.6  348.72  4976.9  348.22  4980.4  348.22
  4980.6  348.72  4986.6   350.7  5036.6  351.73  5103.6  355.45    5112  356.38
  5120.4  355.75  5134.4  356.13  5148.4   357.3  5209.9  359.69  5223.8  360.89
#Mann= 3 ,-1 , 0
  4680.1     .07       0  4976.6     .05       0  4980.6     .07       0
Bank Sta=4976.6,4980.6
XS Rating Curve= 0 ,0
Exp/Cntr=0.3,0.1

Type RM Length L Ch R = 1 ,29252   ,452,452,452
BEGIN DESCRIPTION:
EAST TINSLEY CREEK 57.0
END DESCRIPTION:
XS GIS Cut Line= 3
      2483825.03     13772825.03        2483525.       13772575.
      2483325.01       13772625.
#Sta/Elev= 30
  4614.3  358.76  4635.8  358.36  4692.4  355.98  4734.7  355.16  4756.9  353.82
  4763.4   354.3  4770.5  353.46  4784.2  353.52    4792  352.95  4798.5  353.27
  4905.3  348.03  4919.6  348.87  4926.8  348.56  4948.2  348.83  4969.1  347.72
  4976.9  346.13  4981.4  345.84  4981.6  345.34  4985.1  345.34  4985.4  345.84
  4991.2   347.1  5001.6  348.39  5015.2  348.48  5022.9  350.07    5028  349.87
  5056.4  351.78  5069.3  352.22  5087.3     352  5118.2  353.78    5211  356.58
#Mann= 3 ,-1 , 0
  4614.3     .07       0  4981.4     .05       0  4985.4     .07       0
Bank Sta=4981.4,4985.4
XS Rating Curve= 0 ,0
Exp/Cntr=0.3,0.1

Type RM Length L Ch R = 1 ,28800   ,476,476,476
BEGIN DESCRIPTION:
EAST TINSLEY CREEK 56.0
END DESCRIPTION:
XS GIS Cut Line= 3
      2483925.02     13772625.02        2483425.       13772225.
      2483225.04       13772225.
#Sta/Elev= 30
  4359.5   357.1  4401.9  356.59    4410  355.71  4430.8   355.7    4466   353.9
    4602  351.19  4701.3  350.58  4715.7  351.21  4736.5  350.59  4750.9  351.31
  4757.3  350.63  4807.7   350.3  4858.2  347.93  4914.2  346.86  4922.2  346.38
  4928.6   344.9  4949.4  345.18  4957.4  346.12  4963.8  345.08  4992.6   346.1
  5012.5  345.09  5019.8  344.84  5027.8  342.69  5028.1  342.19  5031.8  342.69
  5049.8  346.53  5059.3  346.91  5099.8  348.69  5169.8  355.36  5199.8  357.03
#Mann= 5 ,-1 , 0
  4359.5     .07       0  5012.5     .12       0  5027.8     .05       0
  5031.8     .12       0  5059.3     .07       0
Bank Sta=5027.8,5031.8
XS Rating Curve= 0 ,0
Exp/Cntr=0.3,0.1

Type RM Length L Ch R = 1 ,28324   ,464,464,464
BEGIN DESCRIPTION:
EAST TINSLEY CREEK 55.0
END DESCRIPTION:
XS GIS Cut Line= 3
      2484025.02     13772475.04        2483725.       13771925.
       2483155.3     13771616.31
#Sta/Elev= 30
  4373.7   355.9  4419.3  355.21  4476.3  352.59  4550.8  350.42  4594.4  350.45
  4624.3  349.26  4647.1   349.9  4654.3   349.1  4749.6  348.01  4779.5  348.25
  4841.9  346.58  4926.7  344.97  4955.8  343.69  4964.7  344.51  4986.5  343.44
  4990.2  340.77  4990.4  340.27  4994.2  340.77  5003.1  340.79  5008.3  343.27
  5045.7  344.54  5057.8   346.2  5073.9  346.19  5170.9  350.31  5183.3  351.45
  5215.7  351.78  5443.8  361.45  5494.3  362.74  5554.2  366.01  5648.2  369.09
#Mann= 5 ,-1 , 0
  4373.7     .07       0  4841.9    .035       0  4955.8     .07       0
  4990.2     .05       0  4994.2     .07       0
Bank Sta=4990.2,4994.2
XS Rating Curve= 0 ,0
Exp/Cntr=0.3,0.1

Type RM Length L Ch R = 1 ,27860   ,453,453,453
BEGIN DESCRIPTION:
EAST TINSLEY CREEK 54.0
END DESCRIPTION:
XS GIS Cut Line= 3
      2484825.02     13771925.01        2484025.       13771725.
        2483225.       13771475.
#Sta/Elev= 30
  4175.7  363.48  4482.4  350.29  4729.8   345.8  4783.9  346.11  4812.2  343.19
  4819.3  343.67  4853.5  341.31  4858.6  342.53  4876.7  340.56  4894.7  343.39
  4899.8  340.06  4953.8  340.19  4977.2   338.8  4982.3  342.01  4995.5  338.08
  4995.8  337.58    5000  338.08    5003  338.08  5010.8  341.61  5016.6  342.08
    5097  343.36  5157.5  346.25  5346.1  349.75  5357.1  351.07  5389.6  349.74
  5416.8  352.05    5422   350.7  5461.3  353.46  5670.9  362.23  5838.5  371.95
#Mann= 6 ,-1 , 0
  4175.7     .07       0  4819.3    .035       0  4953.8     .12       0
  4995.5     .05       0    5000     .12       0    5097     .07       0
Bank Sta=4995.5,5000
XS Rating Curve= 0 ,0
Exp/Cntr=0.3,0.1

Type RM Length L Ch R = 1 ,27407   ,394,394,394
BEGIN DESCRIPTION:
EAST TINSLEY CREEK 53.0
END DESCRIPTION:
XS GIS Cut Line= 3
        2484975.       13771875.        2484175.       13771325.
      2483374.98       13771375.
#Sta/Elev= 30
  4025.1  370.13  4182.9  364.11  4226.7  360.77  4420.9  351.67  4543.3  348.79
  4686.7  347.86  4728.8  346.61  4788.5  346.01  4830.2  345.96  4874.6  343.78
  4923.1  343.11  4952.6  340.34  4959.5  337.23  4967.5  338.84  4971.3  336.73
  4971.6  336.23  4975.8  336.73  4982.4  339.71  4988.5  337.34  4992.9  340.15
  5005.9  341.29    5057  341.37  5166.3  341.07  5246.4  344.05  5276.5  343.45
  5346.6  346.18  5456.8  348.39  5617.1   354.3  5737.4  360.05  5797.5  364.07
#Mann= 6 ,-1 , 0
  4025.1     .07       0  4728.8    .035       0  4788.5     .12       0
  4971.3     .05       0  4975.8     .12       0    5057     .07       0
Bank Sta=4971.3,4975.8
XS Rating Curve= 0 ,0
Exp/Cntr=0.3,0.1

Type RM Length L Ch R = 1 ,27013   ,521,521,521
BEGIN DESCRIPTION:
X19089
END DESCRIPTION:
XS GIS Cut Line= 3
      2485003.03     13771092.69      2484061.53     13770981.93
      2483341.61     13771218.55
#Sta/Elev= 30
    3910  355.53  3928.1   355.7  3938.2  354.89  3978.5  354.52  4018.9  353.06
    4137  349.64  4169.8   349.4  4210.1  347.57  4358.5  344.96  4572.6  343.74
  4823.3  343.39  4951.1   342.6  4977.7  340.81  4999.5  335.69  4999.8  335.19
    5004  335.69  5009.5  336.28  5014.7  338.95  5022.8  339.81  5041.3  339.91
  5073.1  338.53  5086.2  339.15  5135.6  340.08  5212.2   345.4  5396.4  352.05
  5443.8  354.79  5454.3  354.52  5523.6  356.91  5592.4  360.34  5615.8  360.44
#Mann= 8 ,-1 , 0
    3910     .07       0  4018.9    .035       0    4137     .07       0
  4823.3     .12       0  4999.5     .05       0    5004     .12       0
  5086.2     .12       0  5135.6     .07       0
Bank Sta=4999.5,5004
XS Rating Curve= 0 ,0
Exp/Cntr=0.3,0.1

Type RM Length L Ch R = 1 ,26492   ,473,473,473
BEGIN DESCRIPTION:
EAST TINSLEY CREEK 52.0
END DESCRIPTION:
XS GIS Cut Line= 3
      2484801.61     13770684.88        2483875.       13770725.
      2483230.82     13770981.92
#Sta/Elev= 30
  4073.4  349.17  4147.9  348.46  4193.4  348.33  4230.2  346.49  4320.2  344.89
  4840.1  340.26  4860.7  340.12  4880.5  341.87  4885.5  339.56  4890.8  338.94
  4900.8  340.51  4910.8  340.49  4930.8  337.43  4980.9  338.22  4988.6  334.02
  4988.9  333.52  4993.2  334.02  4998.4     337  5003.6     337  5010.3  339.02
  5054.7  338.87    5117  342.33  5162.4  343.54  5194.7  342.42    5261  344.45
  5309.5  344.41  5339.2  345.23  5345.4  346.27    5453  347.64  5694.4  353.08
#Mann= 6 ,-1 , 0
  4073.4     .12       0  4147.9     .07       0  4840.1     .12       0
  4988.6     .05       0  4993.2     .12       0    5117     .07       0
Bank Sta=4988.6,4993.2
XS Rating Curve= 0 ,0
Exp/Cntr=0.3,0.1

Type RM Length L Ch R = 1 ,26019   ,453,453,453
BEGIN DESCRIPTION:
EAST TINSLEY CREEK 51.0
END DESCRIPTION:
XS GIS Cut Line= 3
      2485074.98     13769725.01        2483875.       13770325.
      2483274.97     13770875.03
#Sta/Elev= 30
  3654.3  359.08  3991.4  348.04  4089.9  344.55  4094.9  344.21  4115.5  343.51
  4123.9  340.79  4137.8  343.26    4519  343.09  4551.9  342.64    4879     336
  4942.8  337.71  4987.8  336.58  5009.8  332.32  5031.4  336.48  5066.5  336.86
  5073.9  335.22  5083.1   336.6  5102.3   335.4  5106.8  332.23  5107.1  331.73
  5111.4  332.23  5123.3  335.43  5130.7  332.41  5137.4  332.36  5144.8  336.71
  5151.6  335.36  5158.7  337.28  5236.7   341.8  5363.7  340.14  5809.9  349.26
#Mann= 11 ,-1 , 0
  3654.3     .07       0  3991.4     .12       0  4089.9     .07       0
  4094.9     .12       0    4519     .07       0  4551.9     .12       0
    4879     .07       0  4987.8     .12       0  5083.1     .07       0
  5106.8     .05       0  5111.4     .07       0
Bank Sta=5106.8,5111.4
XS Rating Curve= 0 ,0
Exp/Cntr=0.3,0.1

Type RM Length L Ch R = 1 ,25566   ,466,466,466
BEGIN DESCRIPTION:
EAST TINSLEY CREEK 50.0
END DESCRIPTION:
XS GIS Cut Line= 3
      2484725.05     13769674.99        2483925.       13769925.
      2483274.99     13770725.02
#Sta/Elev= 30
    4157  349.61  4378.6  343.39  4405.9  341.55  4411.1  339.41  4429.4  337.59
  4443.6  340.84  4529.8  342.27    4817  339.45  4900.9  334.39  4908.8  333.61
  4911.7  331.15    4912  330.65  4916.4  331.15  4924.8  333.42  4953.3   335.1
  5045.5   334.6  5066.3  334.32  5080.7  331.99  5087.1  335.06  5203.7  339.21
  5214.3  339.46  5336.4  340.01  5365.5   337.3    5386  338.04  5407.5  335.29
  5485.1  340.37  5528.2  339.35  5627.3  341.65  5833.5  342.88    6026  346.63
#Mann= 9 ,-1 , 0
    4157     .07       0  4529.8     .12       0    4817     .07       0
  4911.7     .05       0  4916.4     .07       0  4924.8     .12       0
  5203.7     .07       0  5214.3     .12       0  5365.5     .07       0
Bank Sta=4911.7,4916.4
XS Rating Curve= 0 ,0
Exp/Cntr=0.3,0.1

Type RM Length L Ch R = 1 ,25100   ,435,435,435
BEGIN DESCRIPTION:
EAST TINSLEY CREEK 49.0
END DESCRIPTION:
XS GIS Cut Line= 3
      2484825.02       13769625.        2483625.       13769625.
      2482825.05     13769724.99
#Sta/Elev= 30
  3799.7  353.29  4229.7  339.75  4294.5  340.07  4325.7  337.52  4389.7  340.42
  4595.8  338.72  4789.7  336.44  4909.7  332.55  4989.7  332.99  5027.6  328.72
    5028  328.22  5032.3  328.72  5042.6  331.72  5050.1  329.05  5080.3  333.28
  5130.7   335.3  5219.6  335.36  5271.8  329.82  5279.4  332.34  5322.2  334.73
  5332.3  331.31  5352.4  334.64  5372.6  335.01  5412.9  330.86  5433.1  334.92
  5453.2  335.97  5503.6   332.1  5521.3  336.18    5554   338.5  5805.9  347.29
#Mann= 7 ,-1 , 0
  3799.7     .07       0  4294.5     .12       0  4325.7     .07       0
  4595.8     .12       0  5027.6     .05       0  5032.3     .12       0
  5219.6     .07       0
Bank Sta=5027.6,5032.3
XS Rating Curve= 0 ,0
Exp/Cntr=0.3,0.1

Type RM Length L Ch R = 1 ,24665   ,467,467,467
BEGIN DESCRIPTION:
EAST TINSLEY CREEK 48.0
END DESCRIPTION:
XS GIS Cut Line= 3
      2484374.98       13769375.        2483575.       13769275.
      2482774.97       13769325.
#Sta/Elev= 30
  4194.7  342.39  4263.9  341.14  4393.7  337.68  4436.6  338.47  4446.6  335.74
  4466.8  338.83  4859.8  334.73  4900.1  331.92  4910.2  328.71  4920.3  328.16
  4930.4  330.96  4963.1  330.41  4980.8   331.9    4993  330.95  5007.4  330.92
  5078.6  330.92  5171.2  334.21  5201.3  333.91  5251.4  330.05  5261.4  330.69
    5269  328.07  5269.3  327.57  5273.9  328.07  5281.5  331.17  5291.5  332.38
  5311.5  332.06  5381.7  336.04  5632.1  341.86  5724.8  345.77  5802.5  347.24
#Mann= 6 ,-1 , 0
  4194.7     .12       0  4263.9     .07       0    4993     .12       0
  5007.4     .07       0    5269     .05       0  5273.9     .07       0
Bank Sta=5269,5273.9
XS Rating Curve= 0 ,0
Exp/Cntr=0.3,0.1

Type RM Length L Ch R = 1 ,24198   ,477,477,477
BEGIN DESCRIPTION:
EAST TINSLEY CREEK 47.0
END DESCRIPTION:
XS GIS Cut Line= 3
      2484474.99     13768375.01        2483275.       13768975.
      2482925.04     13769224.97
#Sta/Elev= 30
  3664.3  348.54  3812.4  342.87  3851.6  340.42    4101  335.41  4164.6  334.31
  4245.7   335.8  4416.2  334.56  4617.4  335.01  4688.6  332.49  4723.6  329.72
  4751.6  330.69  4849.4  328.98  4888.9  329.69  4952.8  330.67  4969.6  329.55
  4972.4  326.46  4972.9  325.96  4977.9  326.46    4992  328.38  4997.5  330.24
  5003.1  328.59  5034.2  330.41  5055.1  329.88  5063.7  330.32  5069.8  331.93
  5078.4  331.54  5084.6  332.74  5128.8  334.86  5286.1  337.02    5436  341.83
#Mann= 6 ,-1 , 0
  3664.3     .07       0    4101     .12       0  4688.6     .07       0
  4888.9     .12       0  4972.4     .05       0  4977.9     .07       0
Bank Sta=4972.4,4977.9
XS Rating Curve= 0 ,0
Exp/Cntr=0.3,0.1

Type RM Length L Ch R = 1 ,23721   ,477,477,477
BEGIN DESCRIPTION:
EAST TINSLEY CREEK 46.0
END DESCRIPTION:
XS GIS Cut Line= 3
      2484275.01       13768275.        2483075.       13768575.
      2482725.05     13768674.99
#Sta/Elev= 30
  3763.3  341.28  3856.1  337.41  3955.9  334.58  3992.7  333.94  4028.7  331.35
  4033.9  332.77  4041.6  331.38  4062.2  333.85  4087.2  334.48  4194.2  333.52
  4474.5  333.55  4482.3  332.37  4487.4  333.44  4505.5  333.84  4612.3  333.41
  4749.8  333.35  4866.2  331.93    4977  328.45  4982.2  327.92  4987.2  323.44
  4987.6  322.94  4992.7  323.44  5010.6  326.17  5017.1   325.1  5027.8  325.48
  5041.8  325.08  5050.9  328.03  5062.6  327.84  5114.6  330.59  5364.2  338.74
#Mann= 9 ,-1 , 0
  3763.3     .07       0  3955.9     .12       0  4087.2     .07       0
  4194.2     .12       0  4612.3     .07       0  4749.8     .12       0
  4987.2     .05       0  4992.7     .12       0  5027.8     .07       0
Bank Sta=4987.2,4992.7
XS Rating Curve= 0 ,0
Exp/Cntr=0.3,0.1

Type RM Length L Ch R = 1 ,23244   ,468,468,468
BEGIN DESCRIPTION:
EAST TINSLEY CREEK 45.0
END DESCRIPTION:
XS GIS Cut Line= 3
      2484424.99       13768225.        2482875.       13768175.
      2482574.97     13768475.03
#Sta/Elev= 30
  3453.4  347.09  3633.5  339.44  3788.5  334.25  3873.6  332.77  3913.6   330.2
  3933.6  329.89  3943.6  330.22  3953.7  332.57  3963.7  333.23  4203.8  332.82
  4213.8     332  4574.2  331.98    4694  331.72  4775.2   330.3  4854.1  328.24
  4894.1  324.39  4914.2  326.88  4955.2   327.8  4984.2  328.34  4994.2  326.87
  4998.9  322.35  4999.3  321.85  5004.5  322.35  5021.5   325.3  5037.2     327
  5046.6  329.43  5060.8  329.25  5117.3   332.1  5173.9   332.5  5428.5  338.63
#Mann= 9 ,-1 , 0
  3453.4     .07       0  3788.5     .12       0  4574.2     .07       0
  4775.2     .12       0  4955.2     .15       0  4998.9     .05       0
  5004.5     .15       0  5021.5     .12       0  5037.2     .07       0
Bank Sta=4998.9,5004.5
XS Rating Curve= 0 ,0
Exp/Cntr=0.3,0.1

Type RM Length L Ch R = 1 ,22776   ,475,475,475
BEGIN DESCRIPTION:
EAST TINSLEY CREEK 44.0
END DESCRIPTION:
XS GIS Cut Line= 3
      2484174.98       13768075.        2482975.       13767775.
      2482524.98       13767825.
#Sta/Elev= 30
    3763  337.07  3845.7  334.47  3963.9  331.72  3979.4  331.08  3987.2  328.48
  4010.4  328.99  4028.4  331.32  4051.6  332.17  4267.7  331.49  4453.6  331.75
  4487.1  329.56  4515.5   331.5  4608.7  331.24    4738  330.35  4886.5  328.28
  4935.5  325.25  4948.4  325.82  4958.7  324.39  4976.7  325.49  4989.6  322.88
  4994.3  320.65  4994.8  320.15  5000.4  320.65  5002.4  320.65    5010  325.59
    5020  326.18  5090.5  326.32  5160.9  330.04  5203.4  330.87  5452.7  336.02
#Mann= 9 ,-1 , 0
    3763     .07       0  3845.7     .12       0  3963.9     .07       0
  4267.7     .12       0  4608.7     .07       0    4738     .12       0
  4994.3     .05       0  5000.4     .12       0  5203.4     .07       0
Bank Sta=4994.3,5000.4
XS Rating Curve= 0 ,0
Exp/Cntr=0.3,0.1

Type RM Length L Ch R = 1 ,22301   ,445,445,445
BEGIN DESCRIPTION:
EAST TINSLEY CREEK 43.0
END DESCRIPTION:
XS GIS Cut Line= 3
      2484288.08      13767744.6        2482925.       13767375.
      2482163.47     13767492.86
#Sta/Elev= 30
  3588.5  340.26  3623.6  338.78  3710.9  336.22  3875.9  331.57  4057.9  328.39
  4078.7  325.93  4093.2  328.51  4204.6  328.16  4234.1  330.02  4257.8  328.81
  4292.5  329.84  4327.1  327.85  4399.9  330.18  4487.1  329.65  4678.6  329.62
  4928.3   327.2  4983.5  323.82  4987.3  319.63  4987.8  319.13  4993.5  319.63
  5003.3  320.93  5010.9  323.93    5050  325.05  5081.8  325.11  5097.9  322.14
  5112.1  324.73  5253.8   330.4  5516.9  335.66  5607.9  339.21  5771.4  339.57
#Mann= 11 ,-1 , 0
  3588.5     .07       0  3623.6     .05       0  3710.9     .07       0
  3875.9     .12       0  4093.2     .07       0  4204.6     .12       0
  4487.1     .07       0  4678.6     .12       0  4987.3     .05       0
  4993.5     .12       0    5050     .07       0
Bank Sta=4987.3,4993.5
XS Rating Curve= 0 ,0
Exp/Cntr=0.3,0.1

Type RM Length L Ch R = 1 ,21856   ,446,446,446
BEGIN DESCRIPTION:
EAST TINSLEY CREEK 42.0
END DESCRIPTION:
XS GIS Cut Line= 3
      2484174.96     13767574.98        2482975.       13766975.
      2482475.01       13767125.
#Sta/Elev= 30
  3650.4  335.77  3685.6  334.49  3803.2  331.85  3883.7  330.48  3950.5  329.73
  3992.3  329.97  4066.8  328.56  4133.9  324.17  4150.7  326.64    4187  327.13
  4240.1  325.15  4245.7  322.86  4262.5  325.36  4312.8  325.61  4329.6   328.2
  4410.6  325.86  4482.3   327.4  4769.4  328.35  4961.3  325.72  4983.6  323.37
  4986.1  318.89  4986.6  318.39  4992.3  318.89  5033.8  324.09  5151.2   323.9
  5169.5  320.14  5184.3   323.5  5255.6  324.16    5347   329.9    5514  334.49
#Mann= 10 ,-1 , 0
  3650.4     .05       0  3685.6     .07       0  3803.2     .05       0
  3883.7     .07       0  3950.5     .05       0  3992.3     .12       0
  4482.3     .07       0  4769.4     .12       0  4986.1     .05       0
  4992.3     .12       0
Bank Sta=4986.1,4992.3
XS Rating Curve= 0 ,0
Exp/Cntr=0.3,0.1

Type RM Length L Ch R = 1 ,21410   ,419,419,419
BEGIN DESCRIPTION:
EAST TINSLEY CREEK 41.0
END DESCRIPTION:
XS GIS Cut Line= 3
      2484325.02     13767375.01        2482775.       13766725.
      2482424.99       13766725.
#Sta/Elev= 30
  3318.7  337.68  3557.3  332.43  3805.7   329.7  3911.3  329.03  3922.3  329.01
  4016.8  328.46  4182.9  328.15  4258.3  324.51  4283.4  324.11  4288.8  322.66
  4294.7  324.19  4312.6  324.27  4327.2  321.98  4330.5  322.72  4348.9   325.3
  4394.7   326.9  4717.6  326.56  4793.5  323.42  4955.7  323.27  4961.1  321.28
  4984.9   320.6  4990.3  321.63  4993.6  317.94  4994.1  317.44  4999.9  317.94
  5019.5  322.85  5059.5  325.19  5149.5  329.15  5169.5   328.6  5349.5  334.67
#Mann= 9 ,-1 , 0
  3318.7     .05       0  3805.7     .07       0  3911.3     .12       0
  3922.3     .07       0  4016.8     .12       0  4258.3     .07       0
  4330.5     .12       0  4993.6     .05       0  4999.9     .12       0
Bank Sta=4993.6,4999.9
XS Rating Curve= 0 ,0
Exp/Cntr=0.3,0.1

Type RM Length L Ch R = 1 ,20991   ,442,442,442
BEGIN DESCRIPTION:
EAST TINSLEY CREEK 40.0
END DESCRIPTION:
XS GIS Cut Line= 3
      2483974.99       13766925.        2482975.       13766525.
      2482725.02     13766225.03
#Sta/Elev= 30
  3922.9   330.8  4380.1  326.32  4515.3  324.77    4644  324.53  4698.4   324.2
  4715.9  322.57  4740.1  322.15  4745.5  323.11    4763  321.59  4769.7  323.78
  4775.1  323.36  4799.3  325.07  4931.3  322.55  4946.1  321.17  4978.4  321.75
  4990.5   320.4  4993.9  316.34  4994.4  315.84  5000.5  316.34  5003.2  316.34
  5007.1  319.01  5013.6  321.14  5021.4  322.33  5064.4  321.63  5093.2  322.08
  5134.7   324.5  5305.2  328.85  5340.3  330.76  5354.6  330.24  5390.4  331.54
#Mann= 6 ,-1 , 0
  3922.9     .05       0  4380.1     .07       0    4644     .12       0
  4993.9     .05       0  5000.5     .12       0  5093.2     .07       0
Bank Sta=4993.9,5000.5
XS Rating Curve= 0 ,0
Exp/Cntr=0.3,0.1

Type RM Length L Ch R = 1 ,20549   ,458,458,458
BEGIN DESCRIPTION:
EAST TINSLEY CREEK 39.0
END DESCRIPTION:
XS GIS Cut Line= 3
      2483875.01     13766775.01        2483075.       13766175.
      2482824.97     13766124.99
#Sta/Elev= 30
  3990.5  329.79  4436.2  325.29  4597.8  323.75  4612.4  324.53  4733.2  323.65
  4747.8  324.52  4804.1  323.59    4877  321.74  4912.4  319.23  4933.2  320.27
  4962.4  320.38  4968.6  316.09  4993.1  317.94  5000.7  320.37  5010.9  320.56
  5031.3  316.24  5041.5  318.77  5051.7   319.3  5061.9  318.54    5068   315.5
  5068.5     315  5076.2   315.5  5092.5  320.21  5123.1  324.72  5133.3  323.23
  5143.5  323.26  5163.9  327.61  5174.1  326.99  5194.5  329.11  5245.5  330.96
#Mann= 4 ,-1 , 0
  3990.5     .05       0  4436.2     .07       0    5068     .05       0
  5076.2     .07       0
Bank Sta=5068,5076.2
XS Rating Curve= 0 ,0
Exp/Cntr=0.3,0.1

Type RM Length L Ch R = 1 ,20091   ,418,418,418
BEGIN DESCRIPTION:
EAST TINSLEY CREEK 38.0
END DESCRIPTION:
XS GIS Cut Line= 3
      2484375.02     13766725.02        2483175.       13765825.
      2482975.03       13765825.
#Sta/Elev= 30
  3502.6  337.51  3658.9  334.54  3856.5  329.18  3916.2  325.51  3924.5  327.35
    3977  327.98  4002.6  324.29  4009.9  327.47  4016.2  326.13  4059.9  328.21
  4368.5  324.53  4466.2  323.38  4545.3  320.19  4689.1  322.06  4766.2  318.88
  4824.5  320.27  4845.3  315.93  4866.2  319.76  4902.6  320.73  4945.3  319.59
  4959.9   315.9  4974.5   316.6  4976.7  315.25  4977.2  314.75  4984.9  315.25
  4989.1  317.13  4995.3   316.6  4999.5  319.58  5037.7     324  5202.6  331.09
#Mann= 8 ,-1 , 0
  3502.6     .05       0  3658.9     .07       0  3856.5     .12       0
    3977     .05       0  4368.5     .07       0  4976.7     .05       0
  4984.9     .07       0  5037.7     .05       0
Bank Sta=4976.7,4984.9
XS Rating Curve= 0 ,0
Exp/Cntr=0.3,0.1

Type RM Length L Ch R = 1 ,19673   ,432,432,432
BEGIN DESCRIPTION:
EAST TINSLEY CREEK 37.0
END DESCRIPTION:
XS GIS Cut Line= 3
      2484318.29      13766541.3        2483275.       13765575.
      2482873.36     13765373.26
#Sta/Elev= 30
    3586  334.77  3601.6  334.45  4018.5  326.45  4031.4  326.65  4038.8   322.8
  4129.4  326.21  4505.4  321.25  4555.3  317.54  4590.5  319.49  4604.6  316.08
    4612  319.26  4668.2  321.66  4809.9  320.88  4852.4  316.82  4909.1  318.13
  4923.3  313.19  4930.1  313.29  4937.4  318.17  4951.6  318.79  4982.6  312.83
  4983.1  312.33  4990.9  312.83    5001  318.15  5044.3  313.41  5055.1  319.36
  5060.8  321.79  5083.4  328.87  5105.7  331.42  5381.1  340.53  5457.5  341.33
#Mann= 9 ,-1 , 0
    3586     .05       0  3601.6     .07       0  4018.5     .05       0
  4129.4     .07       0  4982.6     .05       0  4990.9     .07       0
  5055.1     .05       0  5060.8     .07       0  5381.1     .05       0
Bank Sta=4982.6,4990.9
XS Rating Curve= 0 ,0
Exp/Cntr=0.3,0.1

Type RM Length L Ch R = 1 ,19241   ,443,443,443
BEGIN DESCRIPTION:
EAST TINSLEY CREEK 36.0
END DESCRIPTION:
XS GIS Cut Line= 4
      2484283.09     13766239.26        2483625.       13765475.
        2483425.       13765325.       2483230.8     13765179.35
#Sta/Elev= 30
  3987.9  330.48  4113.9  328.63  4212.2  327.32    4260  326.52  4345.4  324.73
  4406.1  324.19  4478.5  325.34  4803.5   320.7  4868.6  319.99  4876.3  319.03
  4890.6  313.15  4904.1   316.6    4918  313.65  4925.7  315.48  4932.3  314.17
  4939.9   318.2  4960.8  316.62  4970.5  309.76    4971  309.26  4979.7  309.76
  4982.7  313.59  4993.1  316.87  5046.4  317.13    5060  314.77  5168.3  322.93
  5203.7  328.05  5254.8  329.94  5361.8  334.53  5418.3  336.17  5489.2  335.16
#Mann= 12 ,-1 , 0
  3987.9     .05       0  4113.9     .12       0  4212.2     .07       0
    4260     .12       0  4345.4     .07       0  4406.1     .12       0
  4478.5     .07       0  4803.5     .12       0  4970.5     .05       0
  4979.7     .12       0  5254.8     .07       0  5361.8     .05       0
Bank Sta=4970.5,4979.7
XS Rating Curve= 0 ,0
Exp/Cntr=0.3,0.1

Type RM Length L Ch R = 1 ,18798   ,470,470,470
BEGIN DESCRIPTION:
EAST TINSLEY CREEK 35.0
END DESCRIPTION:
XS GIS Cut Line= 4
      2484489.47     13766017.68        2483875.       13765275.
        2483675.       13765175.      2483353.92     13765014.46
#Sta/Elev= 30
  4036.2  331.74  4120.1  330.49  4280.4  328.02  4346.9  324.97  4469.9  324.26
  4766.7  322.19  4886.1   318.6  4914.8  315.62  4935.6  315.21  4957.8  309.87
  4964.3  311.06    4974  309.58  4974.5  309.08  4983.2  309.58  4986.5  314.56
    4993  313.37  4996.9  316.04  5001.6  316.04  5047.9  318.46  5089.6  320.53
  5120.3  320.33  5170.6  325.26  5190.8  325.78  5224.5  327.65  5299.2  330.89
  5433.4  332.78  5522.8  332.59  5550.7  328.14  5567.5  330.54  5582.7  329.99
#Mann= 11 ,-1 , 0
  4036.2     .05       0  4120.1     .07       0  4280.4     .05       0
  4469.9     .07       0  4766.7      .1       0    4974     .05       0
  4983.2      .1       0  5001.6     .12       0  5047.9     .07       0
  5190.8     .12       0  5224.5     .07       0
Bank Sta=4974,4983.2
XS Rating Curve= 0 ,0
Exp/Cntr=0.3,0.1

Type RM Length L Ch R = 1 ,18328   ,417,417,417
BEGIN DESCRIPTION:
EAST TINSLEY CREEK 34.0
END DESCRIPTION:
XS GIS Cut Line= 5
      2484737.14     13765387.57        2484575.       13765175.
        2484275.       13765075.        2483925.       13764925.
      2483548.21     13764763.52
#Sta/Elev= 30
  4412.8  332.14  4448.5  331.32  4733.6  322.08  4862.4  317.19  4880.4   316.5
    4891  312.32  4901.5  315.49  4943.7  316.84  4964.8  311.52  4970.6  307.98
  4971.1  307.48  4979.9  307.98  4985.8  315.13  4993.7  315.69  5039.9  314.92
  5204.2  319.42  5551.2  327.07  5562.1  327.03  5591.1  320.62  5620.1  324.85
  5649.2   323.9  5667.3  328.71  5672.7  326.92  5714.4  329.87  5725.3  326.83
  5743.5  328.65  5748.9  327.25    5767  331.15  5772.5  329.17  5787.1  331.64
#Mann= 7 ,-1 , 0
  4412.8    .035       0  4448.5     .05       0  4733.6     .07       0
  4862.4      .1       0  4970.6     .05       0  4979.9      .1       0
  5204.2     .07       0
Bank Sta=4970.6,4979.9
XS Rating Curve= 0 ,0
Exp/Cntr=0.3,0.1

Type RM Length L Ch R = 1 ,17911   ,428,428,428
BEGIN DESCRIPTION:
EAST TINSLEY CREEK 33.0
END DESCRIPTION:
XS GIS Cut Line= 5
      2484745.94     13765256.41        2484625.       13765075.
        2484425.       13764775.        2484125.       13764575.
      2483838.48     13764383.99
#Sta/Elev= 30
  4421.2  333.25  4430.4  333.33  4436.4  332.05  4502.5  329.26  4559.6   325.8
  4574.6   325.8  4722.8  320.75    4806  318.75  4848.1  316.58  4920.2  315.79
  4950.2  314.53  4977.3  314.97  4992.3  314.27  4996.8  311.72  4999.8  311.72
  5002.6  308.12  5003.1  307.62  5011.6  307.62  5012.1  308.12  5028.3  314.86
  5071.9  317.91  5142.2  318.82  5202.6  320.77  5218.3  320.69  5367.9  323.51
  5468.5  326.95  5506.8  327.39  5584.2  329.36  5620.2  329.34  5704.7  331.15
#Mann= 7 ,-1 , 0
  4421.2     .05       0  4722.8      .1       0  5002.6     .05       0
  5012.1      .1       0  5142.2     .05       0  5218.3    .035       0
  5506.8     .07       0
Bank Sta=5002.6,5012.1
XS Rating Curve= 0 ,0
Exp/Cntr=0.3,0.1

Type RM Length L Ch R = 1 ,17483   ,445,445,445
BEGIN DESCRIPTION:
EAST TINSLEY CREEK 32.0
END DESCRIPTION:
XS GIS Cut Line= 4
      2484921.57       13765088.        2484875.       13764925.
        2484775.       13764575.        2484125.       13764375.
#Sta/Elev= 30
    4472  331.29  4590.8  327.44  4852.8  316.56  4910.6  315.38  4949.6  313.06
  4974.3  314.19  4988.6  312.24  4995.1  306.89  5008.1  307.52  5017.1  306.25
  5017.6  305.75  5026.6  306.25  5027.1   309.5  5047.4  313.19  5059.8  314.88
  5092.5  316.57  5141.5  317.77  5223.3  317.37  5228.5  318.15  5246.2  316.11
  5264.9  316.79    5288  316.48  5299.1  318.42  5331.8  317.73  5364.5   319.4
  5452.7  320.47  5554.8  322.17  5608.5  323.83  5643.7  325.74  5685.6     326
#Mann= 8 ,-1 , 0
    4472     .05       0  4852.8      .1       0  5017.1     .05       0
  5026.6      .1       0  5264.9     .07       0  5452.7     .05       0
  5554.8    .035       0  5608.5     .05       0
Bank Sta=5017.1,5026.6
XS Rating Curve= 0 ,0
Exp/Cntr=0.3,0.1

Type RM Length L Ch R = 1 ,17038   ,347,347,347
BEGIN DESCRIPTION:
EAST TINSLEY CREEK 31.0
END DESCRIPTION:
XS GIS Cut Line= 5
      2485487.38     13764545.79        2485275.       13764475.
        2485125.       13764425.        2484425.       13764225.
      2484041.63     13764115.47
#Sta/Elev= 30
  4625.8  327.82  4733.7  326.86  4821.3  324.68  4852.3  323.82  4893.6  321.23
  4923.5  319.48  4955.1  315.45  4965.6  313.11  4986.7  312.84  4996.4  306.18
  5000.1  304.68  5000.6  304.18  5010.2  304.68  5018.2  309.84  5024.7  312.73
  5029.9     314  5091.4  313.58  5111.8  314.81  5321.4  316.23  5327.5  316.28
  5573.3     318  5807.6  320.94  5809.2  320.94  5898.3  321.73  5910.8  322.68
  5932.1  322.63  5954.2  323.92  6010.1  325.04  6058.2  327.31  6134.5  328.05
#Mann= 12 ,-1 , 0
  4625.8     .05       0  4821.3     .12       0  4893.6     .05       0
  4996.4      .1       0  5000.1     .05       0  5010.2      .1       0
  5091.4     .07       0  5321.4     .12       0  5327.5     .07       0
  5807.6     .05       0  5809.2    .035       0  5910.8     .05       0
Bank Sta=5000.1,5010.2
XS Rating Curve= 0 ,0
Exp/Cntr=0.3,0.1

Type RM Length L Ch R = 1 ,16691   ,542,542,542
BEGIN DESCRIPTION:
EAST TINSLEY CREEK 30.0
END DESCRIPTION:
XS GIS Cut Line= 3
      2485760.26     13764450.95      2485263.09     13764126.71
      2484081.54     13763852.94
#Sta/Elev= 30
  4522.3  325.99  4870.3  321.82  4908.7  318.98  4912.5  318.63  4934.5  321.16
  4963.9  319.87  4970.3   318.9    4979  314.92    4985   313.3  4994.1  312.21
  5000.1  312.62  5006.1  310.27  5010.1  304.58  5010.6  304.08  5020.2  304.58
  5024.2  307.41    5030  311.29  5036.3  312.67  5139.2  312.61  5175.5  314.33
  5257.6  315.39  5371.4  315.12  5408.9  313.67  5432.1   315.2    5483  315.76
  5760.6  317.69  5939.9   320.2  6040.3   322.1  6282.3  327.49  6328.7  328.31
#Mann= 10 ,-1 , 0
  4522.3     .05       0  4908.7     .12       0  5010.1     .05       0
  5020.2     .12       0  5024.2      .1       0  5139.2     .12       0
    5483     .07       0  5939.9    .035       0  6040.3     .05       0
  6282.3     .07       0
Bank Sta=5010.1,5020.2
XS Rating Curve= 0 ,0
Exp/Cntr=0.3,0.1

Type RM Length L Ch R = 1 ,16149   ,460,460,460
BEGIN DESCRIPTION:
EAST TINSLEY CREEK 29.0
END DESCRIPTION:
XS GIS Cut Line= 5
      2485865.94     13764063.09        2485725.       13763975.
        2485325.       13763725.        2484625.       13763775.
      2484283.36      13763799.4
#Sta/Elev= 30
    4370  321.48  4556.4  318.99  4583.7  317.44  4601.7  315.33  4732.5  313.16
  4747.9  312.11  4753.8  314.76  4783.8  311.96  4790.3  314.19  4796.2  312.02
  4826.9   314.9  4848.1  312.31  4884.7  313.21  4890.6  309.92    4900  309.01
  4905.9  311.86  5000.2  310.95  5010.4  308.09  5012.7  303.11  5013.2  302.61
  5023.1  303.11    5028  309.49    5038  313.83  5177.6  313.05  5276.8  313.76
  5375.8  314.69  5474.7  315.81  5573.6  316.88  5771.4  319.89  6052.2  324.17
#Mann= 12 ,-1 , 0
    4370     .05       0  4556.4     .07       0  4583.7     .05       0
  4732.5      .1       0  5012.7     .05       0  5023.1      .1       0
  5177.6     .12       0  5276.8     .07       0  5375.8    .035       0
  5474.7     .07       0  5573.6    .035       0  5771.4     .05       0
Bank Sta=5012.7,5023.1
XS Rating Curve= 0 ,0
Exp/Cntr=0.3,0.1

Type RM Length L Ch R = 1 ,15689   ,461,461,461
BEGIN DESCRIPTION:
EAST TINSLEY CREEK 28.0
END DESCRIPTION:
XS GIS Cut Line= 5
      2485939.05     13763889.05        2485775.       13763725.
        2485375.       13763325.        2484725.       13763325.
      2484593.99       13763325.
#Sta/Elev= 30
  4201.5   321.8    4249  321.42  4292.1  321.12  4337.2  319.72    4430  318.61
  4461.8  318.93  4493.2   317.5  4546.6  317.23  4673.9  312.14  4716.3  311.44
  4815.3  311.11  4942.6  311.86  4970.9  311.19  5001.7  308.77  5003.9  303.33
  5004.4  302.83  5014.4  303.33  5019.2  303.58  5029.2   308.6  5039.2  312.24
  5059.3  312.59  5099.2  311.57  5119.2  313.09  5129.2  312.54  5169.2  313.61
  5289.2  314.26  5409.2  316.13  5539.2  316.67  5701.4  318.54  5780.2  320.27
#Mann= 8 ,-1 , 0
  4201.5     .05       0    4249     .12       0  4337.2     .05       0
  4493.2      .1       0  5003.9     .05       0  5014.4      .1       0
  5059.3     .07       0  5701.4    .035       0
Bank Sta=5003.9,5014.4
XS Rating Curve= 0 ,0
Exp/Cntr=0.3,0.1

Type RM Length L Ch R = 1 ,15228   ,440,440,440
BEGIN DESCRIPTION:
EAST TINSLEY CREEK 27.0
END DESCRIPTION:
XS GIS Cut Line= 5
      2486216.97     13763147.99        2485925.       13763075.
        2485525.       13762975.        2484975.       13763075.
      2484628.17     13763138.06
#Sta/Elev= 30
  4291.6  325.52  4499.8  322.18  4656.4  316.03  4829.6  308.45  4953.3  312.71
  4973.9  309.53  4986.8  305.68  4994.6   305.4  4996.8   300.8  4997.3   300.3
  5007.8   300.8    5015  309.37  5025.2  309.92    5076  308.21  5084.9  310.42
    5090  309.03  5106.5  310.17    5137  307.09  5143.4  309.17  5347.9  312.55
  5360.4   312.6  5402.5   313.2  5595.6  316.82    5635   316.7    5649  315.15
  5746.8  316.25  5767.2  314.84  5828.1  318.26    5895  319.83  5916.4  319.93
#Mann= 8 ,-1 , 0
  4291.6     .07       0  4656.4      .1       0  4996.8     .05       0
  5007.8      .1       0  5347.9     .07       0  5360.4     .05       0
  5402.5      .1       0    5895     .07       0
Bank Sta=4996.8,5007.8
XS Rating Curve= 0 ,0
Exp/Cntr=0.3,0.1

Type RM Length L Ch R = 1 ,14788   ,488,488,488
BEGIN DESCRIPTION:
EAST TINSLEY CREEK 26.0
END DESCRIPTION:
XS GIS Cut Line= 4
      2486174.98       13762575.        2485375.       13762625.
        2485075.       13762725.      2484674.91     13762858.36
#Sta/Elev= 30
    4214  322.78  4215.9  322.78  4429.6  315.89  4451.9  315.37    4457  316.22
  4514.6  314.53  4674.9  312.71  4777.6  309.17  4785.1  309.58    4804  309.03
  4845.2  308.16  4885.3  309.38  4905.3  309.27  4925.4  307.43  4945.4  309.33
  4995.5  307.42  5026.1  307.22  5052.1  299.55  5052.6  299.05  5062.8  299.05
  5063.3  299.55  5068.2   307.6  5078.8  308.81    5142  311.19    5231  313.09
  5279.1  313.42  5458.3  316.76  5484.3  316.52  5718.4  318.79  5753.5  319.63
#Mann= 9 ,-1 , 0
    4214     .05       0  4215.9    .035       0  4429.6     .07       0
    4804      .1       0  5052.1     .05       0  5063.3      .1       0
    5231     .07       0  5484.3     .05       0  5718.4     .07       0
Bank Sta=5052.1,5063.3
XS Rating Curve= 0 ,0
Exp/Cntr=0.3,0.1

Type RM Length L Ch R = 1 ,14300   ,464,464,464
BEGIN DESCRIPTION:
EAST TINSLEY CREEK 25.0
END DESCRIPTION:
XS GIS Cut Line= 4
      2486074.98     13762474.99        2485275.       13762225.
        2485075.       13762175.      2484805.09     13762107.52
#Sta/Elev= 30
  4161.3   318.6  4182.8   318.4    4196  317.41  4339.4   313.5  4415.3  313.06
    4518  311.07    4528  311.46  4611.7  309.32  4674.6  308.15  4680.4  307.52
    4848  305.32  4936.6   307.9  4950.7  306.34  4951.9  298.64  4952.4  298.14
  4962.7  298.14  4963.2  298.64    4978  300.93    4989  306.86    5051  307.93
  5058.7  309.43  5063.9  308.36  5092.2  308.86  5127.3  311.24  5228.8   316.8
  5393.7  321.56  5463.3  324.64  5476.2  325.57  5481.3  327.36  5483.8  327.36
#Mann= 6 ,-1 , 0
  4161.3    .035       0    4196     .07       0  4611.7      .1       0
  4951.9     .05       0  4963.2      .1       0  5127.3     .07       0
Bank Sta=4951.9,4963.2
XS Rating Curve= 0 ,0
Exp/Cntr=0.3,0.1

Type RM Length L Ch R = 1 ,13836   ,863,863,863
BEGIN DESCRIPTION:
EAST TINSLEY CREEK 24.0
END DESCRIPTION:
XS GIS Cut Line= 4
        2486175.       13762425.        2485375.       13761925.
        2485075.       13761925.       2484838.4       13761925.
#Sta/Elev= 30
    4052   321.9  4095.5  320.53  4141.2  318.83  4181.7     317  4327.4  314.42
  4370.4  312.72  4379.2  313.08    4437  310.26  4473.6  310.54  4500.7  309.31
  4531.4  309.64  4671.6  307.39    4720  306.11  4762.5  306.43  4799.1  304.63
  4878.1  306.23  4966.5  306.47  4972.4   305.7  4982.1  298.44  4982.6  297.94
  4993.4  298.44  4995.4  301.42  4997.9  301.42  5005.8  306.34  5045.4  309.72
  5185.4  311.77  5385.4  316.48  5405.4  317.59  5485.4  318.66    5532  320.36
#Mann= 7 ,-1 , 0
    4052     .07       0  4095.5    .035       0  4141.2     .07       0
  4671.6      .1       0  4982.1     .05       0  4993.4      .1       0
  5005.8     .07       0
Bank Sta=4982.1,4993.4
XS Rating Curve= 0 ,0
Exp/Cntr=0.3,0.1

Type RM Length L Ch R = 1 ,12973   ,430,430,430
BEGIN DESCRIPTION:
EAST TINSLEY CREEK 23.0
END DESCRIPTION:
XS GIS Cut Line= 5
      2486257.34      13761827.1        2486075.       13761775.
        2485725.       13761675.      2485455.18     13761472.63
      2484992.94     13761290.08
#Sta/Elev= 30
  4445.8  319.34  4561.7  314.57  4657.5  311.79  4691.3     310  4704.9  304.95
  4718.6  302.52  4725.1  300.33  4739.4  302.96  4812.2  305.46  4831.7  305.28
  4875.9  302.95  4895.4  304.28  4977.3  305.33    5013  303.16  5021.3  299.99
  5021.9  295.46  5022.4  294.96  5033.2  295.46  5042.2  303.47  5049.4  304.91
  5199.4  305.21  5235.9  308.01  5263.4  308.42  5323.5  307.65  5333.7  309.36
  5358.4  308.86  5426.9  310.37  5648.7  317.56  5721.8  318.19  5833.7  317.43
#Mann= 7 ,-1 , 0
  4445.8     .07       0  4561.7     .12       0  4704.9      .1       0
  5021.9     .05       0  5033.2      .1       0  5263.4    .035       0
  5323.5     .05       0
Bank Sta=5021.9,5033.2
XS Rating Curve= 0 ,0
Exp/Cntr=0.3,0.1

Type RM Length L Ch R = 1 ,12543   ,455,455,455
BEGIN DESCRIPTION:
EAST TINSLEY CREEK 22.0
END DESCRIPTION:
XS GIS Cut Line= 4
      2486257.36     13761724.27        2486125.       13761625.
        2485925.       13761475.      2485224.96     13761274.99
#Sta/Elev= 30
  4584.2  317.91  4674.6  314.89  4832.3     310  4849.6   309.8  4886.1  305.96
  4892.4  303.62  4906.9  302.49  4921.5   302.7  4927.8  304.56  4971.5  302.64
  4977.8  303.17  4986.1   300.4  4990.8  296.49  4991.3  295.99  5002.2  296.49
    5010  299.24  5016.5  304.07  5072.4   303.7  5145.2  305.67  5167.3  304.59
    5196  299.81  5201.2  300.09  5207.6  302.49    5218  304.16    5321  306.98
  5380.6   306.1  5394.9   308.2  5422.6  308.34  5519.7  309.31  5727.7  317.37
#Mann= 7 ,-1 , 0
  4584.2     .07       0  4674.6     .12       0  4832.3      .1       0
  4990.8     .05       0  5002.2      .1       0    5321    .035       0
  5422.6     .05       0
Bank Sta=4990.8,5002.2
XS Rating Curve= 0 ,0
Exp/Cntr=0.3,0.1

Type RM Length L Ch R = 1 ,12088   ,427,427,427
BEGIN DESCRIPTION:
EAST TINSLEY CREEK 21.0
END DESCRIPTION:
XS GIS Cut Line= 3
      2486525.02     13761675.01        2485775.       13761075.
      2485054.14     13761215.95
#Sta/Elev= 30
  4039.2  326.12  4140.9  322.41    4437  311.26  4628.8  306.48    4794  302.92
  4843.6  304.41  4871.6  303.47  4878.8  301.48  4885.2   302.5  4893.2  300.52
  4899.6  301.68  4907.6   299.9  4928.5   303.3  4935.7  302.43  4942.9  297.29
  4949.3  303.16  4957.3  300.65  4963.7  303.75  4971.7  302.87  4978.1   304.2
  5009.9  301.15  5019.8  297.12  5020.3  296.62  5031.2  297.12  5050.6  302.61
  5067.9  302.74  5142.3   303.2  5264.6  308.75  5509.2  314.54  5734.2  315.67
#Mann= 7 ,-1 , 0
  4039.2    .035       0  4140.9     .07       0  4628.8      .1       0
  5019.8     .05       0  5031.2      .1       0  5067.9    .035       0
  5142.3     .05       0
Bank Sta=5019.8,5031.2
XS Rating Curve= 0 ,0
Exp/Cntr=0.3,0.1
