HEC-RAS study MCCOY CREEK.prj: MCCOY CREEK Base Level Engineering

--- MCCOY CREEK.g01 (geometry) --- (continued)

Type RM Length L Ch R = 1 ,58999   ,442,442,442
BEGIN DESCRIPTION:
MCCOY CREEK 78.0
END DESCRIPTION:
XS GIS Cut Line= 3
        2516875.       13661125.        2516275.       13661625.
      2515975.01     13662024.98
#Sta/Elev= 30
    4219  317.86  4232.7  317.91  4297.1  314.07  4332.9  311.02  4347.2  310.84
  4431.8  305.53  4567.2  299.74    4588  297.82  4645.3  295.49  4772.9  291.88
    4851  291.99  4893.9  293.11  4914.8  292.55  4935.6  289.87  4943.4  287.09
  4957.7  283.59    4974  284.61  4986.4  283.65    4990  282.67  4990.1  282.64
  4990.6  282.14  5003.4  282.64  5007.3   282.9  5013.6  286.96  5021.9  288.04
  5028.1  289.98  5036.5  289.93  5042.7   291.1  5136.5  291.96    5500  303.31
#Mann= 5 ,-1 , 0
    4219     .05       0    4974     .07       0    4990     .05       0
  4990.1     .05       0  5003.4     .05       0
Bank Sta=4990.1,5003.4
XS Rating Curve= 0 ,0
Exp/Cntr=0.3,0.1

Type RM Length L Ch R = 1 ,58557   ,456,456,456
BEGIN DESCRIPTION:
MCCOY CREEK 77.0
END DESCRIPTION:
XS GIS Cut Line= 3
      2516724.97     13661075.01        2516125.       13661225.
      2515524.99     13662425.02
#Sta/Elev= 30
  4375.2  311.46  4457.6   306.3  4591.6  300.36    4687  294.77    4806  290.75
  4859.6  289.63  4908.1  291.27  4934.4  291.69  4962.7  290.47  4975.6  288.78
  4991.1  283.23  4996.4  283.23    5001  280.99  5001.5  280.49  5014.3  280.99
    5016  282.13  5024.4  281.69  5046.7  283.54  5052.3  286.89  5060.7  287.38
  5074.7  290.92  5097.1  292.08  5124.1  291.68  5210.7  291.55  5440.8  294.08
  5650.7  298.81  5790.2  302.92  6114.8  315.92  6327.2  322.64  6335.3  322.68
#Mann= 10 ,-1 , 0
  4375.2     .05       0    4806     .07       0  4908.1      .1       0
    5001     .05       0  5014.3      .1       0  5124.1     .07       0
  5210.7     .05       0  5650.7     .07       0  6114.8     .05       0
  6327.2     .07       0
Bank Sta=5001,5014.3
XS Rating Curve= 0 ,0
Exp/Cntr=0.3,0.1

Type RM Length L Ch R = 1 ,58101   ,480,480,480
BEGIN DESCRIPTION:
MCCOY CREEK 76.0
END DESCRIPTION:
XS GIS Cut Line= 3
      2516124.98     13660675.02        2515975.       13660825.
        2515475.       13662025.
#Sta/Elev= 30
  4788.4   304.5  4816.7  302.69  4859.1  298.17  4929.8  293.84  4943.9  291.57
  4972.2  281.08  4977.7   280.1  4979.7  279.74  4980.2  279.24  4993.1  279.74
    4997  282.84  5003.2  282.84  5009.7  285.78  5024.6  287.67  5044.4  289.08
  5139.7   288.7  5213.2  290.28  5318.7  290.95  5418.8  291.26  5635.1   292.5
    5872  294.97  5967.6  297.58  6049.7  300.82  6094.7  301.57  6162.4  305.11
  6185.1  305.62    6209  307.59  6214.4  307.15    6262  308.93  6300.5  311.61
#Mann= 11 ,-1 , 0
  4788.4     .05       0  4977.7     .07       0  4979.7     .05       0
  4993.1     .07       0  5024.6     .05       0  5213.2    .035       0
  5318.7     .07       0  5418.8    .035       0  5635.1     .07       0
  5967.6     .05       0  6162.4     .12       0
Bank Sta=4979.7,4993.1
XS Rating Curve= 0 ,0
Exp/Cntr=0.3,0.1

Type RM Length L Ch R = 1 ,57621   ,471,471,471
BEGIN DESCRIPTION:
MCCOY CREEK 75.0
END DESCRIPTION:
XS GIS Cut Line= 3
      2515874.97     13660525.01        2515525.       13660725.
      2515325.01     13661924.97
#Sta/Elev= 30
  4602.3  301.59  4787.7     292  4867.2  289.01  4916.8  285.05  4932.7     285
    4960  281.03  4969.1  278.02  4969.6  277.52  4982.6  278.02  4987.1  278.69
  4991.7  279.38  4996.5  283.63  4997.5  284.51  5015.5  284.96  5038.3  287.58
  5095.2  287.99    5198  288.12  5342.5  290.93  5350.1  290.23  5451.5   291.2
  5459.1  292.13    5715  292.77  5763.2  294.49  5814.5   294.3  5870.1  295.36
  6015.8  298.35  6161.1  303.21  6181.4  304.56  6188.4  306.07  6221.9  307.01
#Mann= 11 ,-1 , 0
  4602.3     .05       0  4787.7      .1       0  4969.1    .035       0
  4982.6      .1       0  4987.1     .05       0  4996.5    .035       0
  5095.2     .05       0  5814.5     .07       0  5870.1     .05       0
  6015.8     .07       0  6188.4     .12       0
Bank Sta=4969.1,4982.6
XS Rating Curve= 0 ,0
Exp/Cntr=0.3,0.1

Type RM Length L Ch R = 1 ,57150   ,469,469,469
BEGIN DESCRIPTION:
MCCOY CREEK 74.0
END DESCRIPTION:
XS GIS Cut Line= 3
        2515675.       13659925.        2515125.       13660525.
      2514525.04     13660924.97
#Sta/Elev= 30
  4190.3  303.55  4199.2  303.47  4329.5  297.63  4431.1  293.34  4437.9  292.39
  4508.8  290.12  4572.3  288.87  4586.5  289.74  4608.1  288.24  4643.2  287.83
    4801  287.54  4912.1  287.06  4926.2  285.61  4933.6  283.64  4947.8  282.59
  4976.2  282.52    4983  280.17  4989.4  276.41  4989.9  275.91  5004.8  276.41
  5007.2   279.9  5011.7   281.9  5017.8   282.9  5068.8  285.79  5134.9  286.36
    5162  288.26    5276   290.2    5483  292.29  5643.8   295.3  5725.3  297.38
#Mann= 9 ,-1 , 0
  4190.3     .05       0  4199.2    .035       0  4329.5     .05       0
    4801      .1       0  4989.4     .05       0  5004.8      .1       0
    5276     .07       0    5483     .05       0  5643.8     .07       0
Bank Sta=4989.4,5004.8
XS Rating Curve= 0 ,0
Exp/Cntr=0.3,0.1

Type RM Length L Ch R = 1 ,56681   ,409,409,409
BEGIN DESCRIPTION:
MCCOY CREEK 73.0
END DESCRIPTION:
XS GIS Cut Line= 3
      2515975.02     13659524.99        2514775.       13660225.
      2514224.99       13660575.
#Sta/Elev= 30
  3610.7  324.96  3628.3  324.29  3902.2  314.28  4163.6  300.66  4339.3  291.79
  4420.7  289.83  4430.6   289.6  4436.4  290.75  4473.6  288.51  4583.2  286.96
  4769.7  285.28    4781  284.91    4861  286.41  4906.1  285.19  4954.9  280.63
  4986.3  279.76  4997.1  275.92  4999.9  275.91  5000.4  275.41  5015.3  275.91
  5028.8  281.53  5035.5   280.8  5049.9  284.79  5059.2  285.52  5101.6  284.35
  5153.2  286.13  5180.3  288.88  5208.1  289.95  5477.5  296.28  5651.9  303.71
#Mann= 11 ,-1 , 0
  3610.7     .07       0  3628.3     .05       0  4163.6     .07       0
  4339.3     .05       0  4420.7     .07       0  4583.2    .035       0
  4769.7     .05       0    4781      .1       0  4999.9     .05       0
  5015.3      .1       0  5208.1     .07       0
Bank Sta=4999.9,5015.3
XS Rating Curve= 0 ,0
Exp/Cntr=0.3,0.1

Type RM Length L Ch R = 1 ,56272   ,434,434,434
BEGIN DESCRIPTION:
MCCOY CREEK 72.0
END DESCRIPTION:
XS GIS Cut Line= 3
      2515374.98     13659675.01        2514775.       13659875.
      2514174.98     13660425.01
#Sta/Elev= 30
  4352.9  296.92  4563.7  288.01  4677.3  286.03  4827.2  284.85  4879.9  281.96
    4901  282.26  4911.6  284.82  4968.3  282.45  4988.7   281.5  4992.4  279.11
  4999.2  281.49  5006.6   277.3  5013.4  280.71  5020.8  275.78  5027.2  274.66
  5027.7  274.16  5042.7  274.66  5055.9  276.76  5077.5  275.27  5105.9  280.75
  5134.3   281.1    5141  278.35  5155.2  282.96    5162  281.65  5171.8  286.18
  5226.1  286.27  5247.1  281.46  5313.2  287.41  5544.3  292.27  5799.3  302.87
#Mann= 7 ,-1 , 0
  4352.9     .07       0  4677.3     .12       0  4968.3      .1       0
  5027.2     .05       0  5042.7      .1       0  5171.8    .035       0
  5313.2     .07       0
Bank Sta=5027.2,5042.7
XS Rating Curve= 0 ,0
Exp/Cntr=0.3,0.1

Type RM Length L Ch R = 1 ,55838   ,429,429,429
BEGIN DESCRIPTION:
MCCOY CREEK 71.0
END DESCRIPTION:
XS GIS Cut Line= 3
      2515774.97       13659525.        2514575.       13659525.
      2514025.01     13660124.99
#Sta/Elev= 30
  3795.3  317.56  3935.3  311.76  4093.9  303.52  4335.3  291.23  4495.9  286.26
  4635.3  284.27    4862  283.41  4925.3  279.68  4955.3  279.03    4985  273.68
  4985.5  273.18  5000.6  273.68  5009.1  274.03  5030.7  278.73  5051.7  279.94
  5073.3  279.81  5094.2  282.61  5115.8  282.74  5144.2  284.49  5195.2  284.92
  5391.4  288.08  5483.6  290.49  5511.3   289.8  5604.2  291.89  5646.4  294.02
  5653.5  293.05  5702.8  294.95  5731.2  294.13  5781.2  298.91  5809.2  299.55
#Mann= 9 ,-1 , 0
  3795.3     .05       0  4093.9     .07       0  4495.9     .12       0
    4862      .1       0    4985     .05       0  5000.6      .1       0
  5195.2     .07       0  5391.4     .05       0  5511.3     .07       0
Bank Sta=4985,5000.6
XS Rating Curve= 0 ,0
Exp/Cntr=0.3,0.1

Type RM Length L Ch R = 1 ,55409   ,440,440,440
BEGIN DESCRIPTION:
MCCOY CREEK 70.0
END DESCRIPTION:
XS GIS Cut Line= 3
      2515624.99       13658475.        2514425.       13659175.
      2513825.04     13659574.97
#Sta/Elev= 30
  3610.3  327.84  3800.1  320.23  3991.9  308.43  4107.7  300.72  4337.6  288.04
  4473.2  282.86  4598.9  282.24  4819.2  282.32  4895.8     282  4976.4  275.95
  4983.7  273.85  4984.2  273.35  4999.6  273.85  5013.1   276.1  5028.1  274.73
  5043.1  281.21  5058.1  282.12  5064.1  279.67  5094.2  281.36  5151.3  279.19
  5193.3  283.93  5244.4  286.66  5274.5  286.42  5301.5  283.54  5331.5  284.32
  5352.6  287.53  5396.1  287.49  5397.1  287.46  5584.9  292.11  5720.6  294.86
#Mann= 11 ,-1 , 0
  3610.3     .07       0  3991.9     .12       0  4107.7     .07       0
  4337.6      .1       0  4598.9     .12       0  4819.2      .1       0
  4983.7     .05       0  4999.6      .1       0  5396.1     .07       0
  5397.1     .05       0  5584.9     .07       0
Bank Sta=4983.7,4999.6
XS Rating Curve= 0 ,0
Exp/Cntr=0.3,0.1

Type RM Length L Ch R = 1 ,54969   ,430,430,430
BEGIN DESCRIPTION:
MCCOY CREEK 69.0
END DESCRIPTION:
XS GIS Cut Line= 3
      2515475.04     13658474.99        2514375.       13658775.
      2513474.96       13658675.
#Sta/Elev= 30
  3868.2  322.36  3940.8  319.87  4085.9  308.65  4170.5  303.11  4358.6  291.43
  4456.1  286.13  4461.4  285.78  4564.2  281.37  4593.8  280.63  4795.3  280.66
  4842.6  280.82  4869.6  278.62  4877.1  278.68  4911.7  275.41  4916.9  276.14
  4946.2  276.11    4959  274.09  4959.5  273.59    4975  274.09  4991.1  274.92
  5005.8  277.24  5028.5  278.52    5102  280.48  5212.4  283.03  5326.3  284.68
  5441.1  285.92  5500.3  287.81  5537.5  288.38  5722.8   293.8    5914  301.17
#Mann= 15 ,-1 , 0
  3868.2     .07       0  4170.5     .12       0  4358.6     .07       0
  4456.1     .12       0  4461.4     .07       0  4564.2     .05       0
  4795.3     .12       0  4869.6      .1       0    4959     .05       0
    4975      .1       0    5102     .05       0  5212.4     .07       0
  5326.3     .05       0  5500.3     .07       0  5537.5     .05       0
Bank Sta=4959,4975
XS Rating Curve= 0 ,0
Exp/Cntr=0.3,0.1

Type RM Length L Ch R = 1 ,54539   ,456,456,456
BEGIN DESCRIPTION:
MCCOY CREEK 68.0
END DESCRIPTION:
XS GIS Cut Line= 3
      2515074.97     13658125.01        2514475.       13658375.
        2513275.       13658675.
#Sta/Elev= 30
  4349.5  304.62  4441.1  299.26  4464.8   296.7  4647.9  282.36  4739.5  278.58
  4777.9  279.84  4807.2  279.58    4831  278.76  4869.5  274.39  4884.1  275.61
  4916.4   273.8  4945.3  275.25  4947.5  273.65    4948  273.15  4963.6  273.65
  4977.8  275.01  4988.2  274.12  5009.8  274.12  5017.5  276.36  5022.7  274.63
  5030.4  276.63  5058.7  279.73    5100  281.13  5154.1     281  5182.4  279.89
  5257.2  280.12  5677.2  286.92  5834.4  292.61  6030.2  301.12  6236.4  307.35
#Mann= 6 ,-1 , 0
  4349.5     .07       0  4441.1     .05       0  4916.4      .1       0
  4947.5     .05       0  4963.6      .1       0  4988.2     .05       0
Bank Sta=4947.5,4963.6
XS Rating Curve= 0 ,0
Exp/Cntr=0.3,0.1

Type RM Length L Ch R = 1 ,54083   ,431,431,431
BEGIN DESCRIPTION:
MCCOY CREEK 67.0
END DESCRIPTION:
XS GIS Cut Line= 3
      2514825.04     13657924.99        2514525.       13657975.
      2513325.03     13657775.01
#Sta/Elev= 30
  4700.1  290.89  4733.1  289.63  4915.6  278.81  4971.3  273.26    4976  269.47
  4976.5  268.97  4992.1  269.47  5001.7  274.06  5065.1  275.85  5105.7  275.39
  5146.2  277.87  5166.5   275.9  5176.6  275.81  5288.1   278.2  5328.7  277.35
  5389.5  277.75  5430.1  278.91  5584.7  280.66  5706.3  283.54  5876.1  289.49
  5896.4  291.09  5916.7  290.79  5967.4  293.91  5997.8  294.23  6048.5  297.95
  6066.2  297.02  6119.5  299.84  6132.1  301.18  6149.9  300.57  6220.8  304.75
#Mann= 3 ,-1 , 0
  4700.1     .05       0    4976     .05       0  4992.1     .05       0
Bank Sta=4976,4992.1
XS Rating Curve= 0 ,0
Exp/Cntr=0.3,0.1

Type RM Length L Ch R = 1 ,53652   ,434,434,434
BEGIN DESCRIPTION:
MCCOY CREEK 66.0
END DESCRIPTION:
XS GIS Cut Line= 3
      2514925.01       13657825.        2514325.       13657625.
      2513324.96       13657725.
#Sta/Elev= 30
  4367.2  294.27  4535.9  286.58  4641.3   282.7  4757.2  279.86  4883.7  275.52
  4894.3  274.42  4915.3  273.99  4925.9  275.25  4936.4  274.24  4970.4  268.05
  4970.9  267.55  4986.7  268.05    4997  270.56  5001.8  270.56  5009.7  269.69
  5047.4  273.79  5120.3  277.34  5248.4  277.17  5441.9  281.55  5642.9     289
    5663  290.91  5683.1  290.23  5733.3  294.67  5755.9  294.26  5803.7  297.84
  5823.8  297.25  5884.1  301.56  5904.2  300.93  5974.5  304.62  6004.7  304.47
#Mann= 5 ,-1 , 0
  4367.2     .05       0  4757.2     .07       0  4970.4     .05       0
  4986.7     .07       0  5001.8     .05       0
Bank Sta=4970.4,4986.7
XS Rating Curve= 0 ,0
Exp/Cntr=0.3,0.1

Type RM Length L Ch R = 1 ,53218   ,474,474,474
BEGIN DESCRIPTION:
MCCOY CREEK 65.0
END DESCRIPTION:
XS GIS Cut Line= 3
      2514824.96       13657175.        2514225.       13657225.
      2513625.04     13657624.97
#Sta/Elev= 30
    4398  290.29  4428.1  287.94  4448.1  288.81  4498.3  285.57  4518.4  285.97
  4588.6  282.22  4598.7  282.78  4696.5  279.06  4821.9  276.04  4937.3  275.39
  4959.9  269.21  4969.9  269.48  4981.8  267.73  4982.3  267.23  4998.2  267.73
    5000  270.03    5003  270.03  5007.6  272.05  5022.6  273.83  5058.6  272.43
  5085.7  275.28  5136.7  276.47  5202.9  274.63  5446.2  279.87  5504.8  282.31
  5518.3   281.8  5569.4  284.89  5620.5  286.31  5685.1  290.43  5721.1  291.08
#Mann= 3 ,-1 , 0
    4398     .05       0  4981.8     .05       0  4998.2     .05       0
Bank Sta=4981.8,4998.2
XS Rating Curve= 0 ,0
Exp/Cntr=0.3,0.1

Type RM Length L Ch R = 1 ,52744   ,467,467,467
BEGIN DESCRIPTION:
MCCOY CREEK 64.0
END DESCRIPTION:
XS GIS Cut Line= 3
        2515225.       13657125.        2514025.       13656825.
      2513625.04     13656625.02
#Sta/Elev= 30
  3767.2  305.89  3849.7  303.76  3973.4  296.39  3991.4  297.56  4045.6  293.41
  4066.1  294.13  4107.4  291.15    4128  291.73  4189.8  288.12  4210.4  288.63
    4262  285.32  4285.2  286.09  4333.6  283.65  4633.1   275.2  4756.7  273.48
  4839.2  274.18    4932  270.28  4952.6   271.9  4977.8  268.07  4978.3  267.57
  4994.3  268.07  5006.9  268.55  5026.5   276.9  5034.9  278.21  5264.1  287.04
  5347.9  293.13  5361.9  292.79  5392.6  296.47  5406.6  296.14  5451.3  300.21
#Mann= 5 ,-1 , 0
  3767.2     .05       0  4045.6    .035       0  4333.6     .05       0
  4977.8     .05       0  4994.3     .05       0
Bank Sta=4977.8,4994.3
XS Rating Curve= 0 ,0
Exp/Cntr=0.3,0.1

Type RM Length L Ch R = 1 ,52277   ,441,441,441
BEGIN DESCRIPTION:
MCCOY CREEK 63.0
END DESCRIPTION:
XS GIS Cut Line= 3
      2514825.03     13656975.03        2514225.       13656425.
      2513625.05     13656574.99
#Sta/Elev= 30
    4181  287.94  4194.9  288.93    4259   285.2  4293.5  285.62  4357.7  282.33
  4379.3  282.56  4747.4  273.45  4832.2  273.01  4860.2  271.81  4973.7  272.66
  4981.1  270.51  4983.3  267.61  4983.8  267.11  4999.8  267.61  5046.5  268.11
  5054.3  270.33  5059.4  268.78  5067.1  270.05  5100.6  270.03  5170.2  275.96
  5306.8  280.77  5376.4  285.54  5384.1  287.08  5407.3  287.39  5425.3  289.63
  5500.1  293.34  5541.3  296.85  5554.2   296.2  5603.1  300.31  5613.4  299.45
#Mann= 4 ,-1 , 0
    4181    .035       0  4293.5     .05       0  4983.3     .05       0
  4999.8     .05       0
Bank Sta=4983.3,4999.8
XS Rating Curve= 0 ,0
Exp/Cntr=0.3,0.1

Type RM Length L Ch R = 1 ,51836   ,466,466,466
BEGIN DESCRIPTION:
MCCOY CREEK 62.0
END DESCRIPTION:
XS GIS Cut Line= 3
        2514925.       13656625.        2514325.       13656025.
      2513925.03     13655825.02
#Sta/Elev= 30
  4147.6  286.78    4183  286.09    4190  285.18  4218.3  285.65  4245.3  284.04
    4289  282.35  4303.2  282.65  4317.3  281.23  4628.4  273.06    4784  270.52
  4798.1  270.97  4854.7  270.16  4868.8  270.44    4883  271.74  4925.4   272.2
  4967.8   268.5  4996.1  267.56  4996.2  265.95  4996.7  265.45  5012.9  265.95
  5018.5  268.73  5054.8  268.73    5089  271.12    5161  276.83    5189  276.76
  5250.9  279.23  5300.8  281.16  5429.4  288.09    5435  289.02  5443.3  288.53
#Mann= 6 ,-1 , 0
  4147.6    .035       0  4245.3     .05       0  4996.2     .05       0
  5012.9     .05       0    5089     .07       0  5250.9     .05       0
Bank Sta=4996.2,5012.9
XS Rating Curve= 0 ,0
Exp/Cntr=0.3,0.1

Type RM Length L Ch R = 1 ,51370   ,472,472,472
BEGIN DESCRIPTION:
MCCOY CREEK 61.0
END DESCRIPTION:
XS GIS Cut Line= 3
      2515024.98     13656174.98        2514425.       13655625.
      2513824.99       13655575.
#Sta/Elev= 30
  4185.8  287.31  4189.2  287.31  4192.9  285.98  4221.2  286.17  4263.8  282.84
  4298.9  282.61  4335.3  280.68  4546.8  272.94  4661.1  270.29  4782.2  269.11
  4836.9   269.1  4886.6  270.48  4906.5   269.6  4944.5  266.75  4970.1  265.31
  4970.6  264.81  4986.8  265.31  5027.7  268.23  5039.8   270.2    5070  272.86
  5130.2  274.75  5150.2  276.66  5182.8   276.9  5330.9  283.26  5340.9  282.93
  5350.9  283.52    5361  285.66    5371  284.94  5411.1   286.7  5601.8  296.54
#Mann= 9 ,-1 , 0
  4185.8     .05       0  4335.3     .07       0  4661.1    .035       0
  4782.2     .07       0  4906.5    .035       0  4944.5     .07       0
  4970.1     .05       0  4986.8     .07       0  5027.7    .035       0
Bank Sta=4970.1,4986.8
XS Rating Curve= 0 ,0
Exp/Cntr=0.3,0.1

Type RM Length L Ch R = 1 ,50898   ,446,446,446
BEGIN DESCRIPTION:
MCCOY CREEK 60.0
END DESCRIPTION:
XS GIS Cut Line= 3
      2515274.97     13655574.98        2514675.       13655275.
      2514074.96       13655325.
#Sta/Elev= 30
  4329.2   290.4  4365.5  288.67  4538.8  276.61  4719.6   268.2    4740  267.45
    4754   268.5    4768  267.64  4807.1  267.45  4861.6  269.24  4896.6  269.08
  4932.9  267.78  4955.3  268.43  4970.1  267.58  4983.2  262.76  4983.7  262.26
  4999.9  262.76    5000  264.34  5020.1   264.8  5030.1  266.06  5062.7  265.66
  5100.3  266.89  5120.4     269  5240.8  271.29  5418.9  278.52  5431.5  278.91
  5441.5   278.2  5491.7  281.07  5511.8  281.02  5521.8  282.05  5602.1   285.3
#Mann= 6 ,-1 , 0
  4329.2     .05       0  4719.6     .07       0  4861.6      .1       0
  4970.1     .05       0  4983.2     .05       0  4999.9     .05       0
Bank Sta=4983.2,4999.9
XS Rating Curve= 0 ,0
Exp/Cntr=0.3,0.1

Type RM Length L Ch R = 1 ,50452   ,427,427,427
BEGIN DESCRIPTION:
MCCOY CREEK 59.0
END DESCRIPTION:
XS GIS Cut Line= 3
      2515425.02     13655425.02        2514975.       13654975.
      2513974.97     13654574.99
#Sta/Elev= 30
  4359.4   291.1  4387.7  290.36  4797.8  267.48  4896.8  266.19  4925.1  267.38
  4956.8  264.99  4967.5  264.93  4981.7     263  5010.6  263.17  5019.7  261.99
  5020.2  261.49  5036.5  261.99  5040.3  264.64    5082  267.53  5118.3  267.29
  5304.1  271.12  5328.4  270.19  5340.5  271.35  5417.2   272.9    5603  276.14
  5609.7  275.51  5749.8  280.43  5764.6  279.54  5825.1  282.67  5835.9  282.02
  5920.7  285.12  5932.8  284.14  6009.6  287.49  6028.4  286.73  6072.9  288.46
#Mann= 5 ,-1 , 0
  4359.4     .05       0  4956.8     .07       0  5019.7     .05       0
  5036.5     .07       0    5082     .05       0
Bank Sta=5019.7,5036.5
XS Rating Curve= 0 ,0
Exp/Cntr=0.3,0.1

Type RM Length L Ch R = 1 ,50025   ,481,481,481
BEGIN DESCRIPTION:
MCCOY CREEK 58.0
END DESCRIPTION:
XS GIS Cut Line= 3
      2515525.01     13655225.01        2515125.       13654625.
      2514525.01     13653525.02
#Sta/Elev= 30
    4284  287.47  4428.2  281.87  4658.1  270.34  4802.3  265.09  4860.9  264.15
  4868.1  265.11  4925.5  265.78  4940.5   264.6  4953.1   261.2  4953.6   260.7
  4970.1   261.2  4982.6  261.51  4997.6  263.91  5013.2  262.63    5030  262.93
  5078.7  265.52  5138.5  264.87  5278.5  266.51  5335.5  268.94  5536.2   270.4
  5661.5  273.94  5802.5  281.36  5808.5   280.8  5834.7  282.15  5852.3  281.82
  5868.5   285.1  5882.2  286.42  5927.8   287.9  6030.3  294.22  6258.1   301.3
#Mann= 7 ,-1 , 0
    4284     .05       0  4868.1      .1       0  4953.1     .05       0
  4970.1      .1       0    5030     .05       0  5808.5    .035       0
  5834.7     .07       0
Bank Sta=4953.1,4970.1
XS Rating Curve= 0 ,0
Exp/Cntr=0.3,0.1

Type RM Length L Ch R = 1 ,49544   ,320,320,320
BEGIN DESCRIPTION:
B19364
END DESCRIPTION:
XS GIS Cut Line= 3
      2515512.87     13655120.25      2515347.56     13654277.14
      2514570.64     13653406.56
#Sta/Elev= 30
    4032  284.15  4210.6  275.66  4241.2  275.35  4332.9  271.26  4363.6  269.09
  4499.4  266.77  4725.5   264.9  4832.2  264.55  4936.7   262.3  4944.3  263.03
    4951   261.5  4979.4  261.89  4986.9   261.3  4992.5  259.39    4993  258.89
  5009.7  259.39  5014.7  262.21  5030.1  264.26  5135.3   267.1    5277  267.41
  5396.6  270.56  5418.3  272.12  5446.7  272.21  5460.9   274.4  5646.6   283.4
  5758.6  288.61  5793.7  291.79  5850.5  294.93  5967.7     298    6058  300.02
#Mann= 8 ,-1 , 0
    4032     .05       0  4499.4     .07       0  4725.5      .1       0
  4992.5     .05       0  5009.7      .1       0  5030.1     .05       0
  5646.6     .07       0  5967.7     .05       0
Bank Sta=4992.5,5009.7
XS Rating Curve= 0 ,0
Exp/Cntr=0.3,0.1

Type RM Length L Ch R = 1 ,49224   ,702,702,702
BEGIN DESCRIPTION:
MCCOY CREEK 57.0
END DESCRIPTION:
XS GIS Cut Line= 3
      2516306.36     13654431.44      2515656.13     13654117.35
      2514592.68     13653136.55
#Sta/Elev= 30
  4049.3  292.95    4286  283.33  4653.2  264.17  4698.4  263.23  4775.6  263.87
  4816.2  262.71  4844.5  263.11  4866.1  261.83  4917.4  262.33  4949.3  262.91
  4972.1  261.01  4986.3  261.25  4998.7  258.11  4999.2  257.61  5015.9  258.11
  5028.8  261.77  5035.6  262.58  5067.3  263.35    5149  265.34    5170  264.41
  5217.1  265.27  5340.7  267.22  5516.9  272.49    5630  277.92  5678.8  278.79
  5885.1  287.33  5948.6  288.41  6019.5  291.88  6097.2  293.18  6218.1  297.38
#Mann= 10 ,-1 , 0
  4049.3     .05       0  4917.4      .1       0  4949.3    .035       0
  4998.7    .035       0  5015.9    .035       0  5067.3     .05       0
  5217.1      .1       0  5340.7     .12       0  5516.9     .07       0
  5678.8     .05       0
Bank Sta=4998.7,5015.9
XS Rating Curve= 0 ,0
Exp/Cntr=0.3,0.1

Type RM Length L Ch R = 1 ,48522   ,291,291,291
BEGIN DESCRIPTION:
B19362
END DESCRIPTION:
XS GIS Cut Line= 3
      2516256.73     13654249.56      2515926.13      13653665.5
      2515039.53      13652861.5
#Sta/Elev= 30
  4481.6  290.32  4698.8   279.9  4843.3  269.48  4866.2  267.15    4898  266.54
  4941.3  262.59  4958.3  262.13  4984.6  260.44  4991.3  256.23  4991.8  255.73
  5009.6  256.23  5022.1  258.39  5072.9   262.4  5217.7  260.99  5231.9  261.96
  5252.9  260.42    5373  261.62  5486.7  262.76  5515.1  264.57  5543.5  263.73
    5607  266.06  5627.9  265.09  5684.7  266.14  5833.4  271.91  5869.2  272.09
  5953.7  276.36  6059.8  277.01  6095.6  278.84  6244.3  281.57  6349.6  285.64
#Mann= 6 ,-1 , 0
  4481.6     .05       0  4843.3    .035       0  4958.3      .1       0
  4991.3     .05       0  5009.6      .1       0    5373     .05       0
Bank Sta=4991.3,5009.6
XS Rating Curve= 0 ,0
Exp/Cntr=0.3,0.1

Type RM Length L Ch R = 1 ,48231   ,449,449,449
BEGIN DESCRIPTION:
MCCOY CREEK 56.0
END DESCRIPTION:
XS GIS Cut Line= 3
        2516375.     13653874.99        2516225.       13653625.
        2515025.       13652425.
#Sta/Elev= 30
  4704.1  279.66  4740.1   278.8  4754.6  277.14  4762.4  274.55  4820.7  273.61
  4856.9  271.14  4892.6  268.37  4929.6  262.68  4972.3  259.64  4999.2  256.01
  5000.6  254.55  5001.1  254.05  5018.9  254.55  5023.9  256.89  5066.4  260.92
  5151.2  259.58  5260.6   260.5  5266.8  260.55  5398.8  261.51  5402.1  261.47
  5563.2  261.99  5668.1  264.12  5871.9  272.29  5933.5  274.76  6042.2  279.51
  6084.6  279.61  6145.5  283.44  6402.2  295.44  6565.4  304.53  6692.7  316.07
#Mann= 15 ,-1 , 0
  4704.1    .035       0  4740.1     .12       0  4856.9      .1       0
  5000.6     .05       0  5018.9      .1       0  5260.6     .12       0
  5266.8     .05       0  5398.8     .12       0  5402.1     .05       0
  5563.2     .12       0  5668.1     .05       0  5871.9     .07       0
  5933.5     .05       0  6145.5     .07       0  6402.2     .12       0
Bank Sta=5000.6,5018.9
XS Rating Curve= 0 ,0
Exp/Cntr=0.3,0.1

Type RM Length L Ch R = 1 ,47782   ,459,459,459
BEGIN DESCRIPTION:
B19363
END DESCRIPTION:
XS GIS Cut Line= 3
      2516686.55     13654023.66      2516460.63     13653334.89
      2515789.18     13652690.95
#Sta/Elev= 30
  4087.3  288.61  4268.9  281.83    4296  281.31  4322.2  279.65  4372.7   277.6
  4477.3  273.72  4517.4  272.34  4529.3  271.13  4686.6   266.1  4950.4  259.76
  4964.6   258.7  4971.8  256.91  4978.7  256.86  4990.9  254.63  4991.4  254.13
  5009.3  254.63  5021.2  256.86  5042.3  257.75  5049.5  259.19  5077.8  260.42
  5133.7  259.87  5162.7  259.44  5301.3  263.91  5339.5  266.21  5396.1   268.2
  5417.1  269.94  5424.4  269.52  5572.8  276.58    5580  276.18  5742.5  279.43
#Mann= 10 ,-1 , 0
  4087.3     .05       0  4268.9    .035       0  4322.2     .05       0
  4372.7     .12       0  4477.3     .07       0  4686.6      .1       0
  4990.9     .05       0  5009.3      .1       0  5133.7     .12       0
  5301.3     .05       0
Bank Sta=4990.9,5009.3
XS Rating Curve= 0 ,0
Exp/Cntr=0.3,0.1

Type RM Length L Ch R = 1 ,47323   ,445,445,445
BEGIN DESCRIPTION:
MCCOY CREEK 55.0
END DESCRIPTION:
XS GIS Cut Line= 3
      2516775.01     13654025.03        2516475.       13652825.
        2516275.       13652625.
#Sta/Elev= 30
  3762.8  289.43  3943.4  283.19    3969  283.06  3992.2  280.98  4010.2  281.41
  4040.6  280.07  4142.8  275.78  4385.3  266.09  4449.6  263.04  4556.5   260.6
  4610.6  261.06  4742.1  258.44  4803.9  259.29  4816.8  258.36  4865.8  257.87
  4894.1  258.43  4948.2  256.52    4988  254.03  4988.5  253.53  5006.4  254.03
  5013.9  256.75  5042.2  260.58  5112.9  264.71  5141.2  267.87  5155.3  267.64
  5169.5  269.58  5224.3  273.88  5254.3  275.22  5268.5   277.5  5282.6  276.41
#Mann= 9 ,-1 , 0
  3762.8     .05       0  3943.4    .035       0  4040.6     .07       0
  4142.8     .12       0  4385.3     .07       0  4449.6      .1       0
    4988     .05       0  5006.4      .1       0  5224.3     .12       0
Bank Sta=4988,5006.4
XS Rating Curve= 0 ,0
Exp/Cntr=0.3,0.1

Type RM Length L Ch R = 1 ,46878   ,447,447,447
BEGIN DESCRIPTION:
MCCOY CREEK 54.0
END DESCRIPTION:
XS GIS Cut Line= 3
      2517425.03     13653125.03        2516825.       13652575.
      2516575.04     13652475.01
#Sta/Elev= 30
  4190.9  273.63  4204.8  273.98  4268.9  269.83  4289.9  270.21  4339.9  266.97
  4367.6   267.2  4403.4  264.64  4488.5  261.57  4612.4  258.65  4651.2  257.79
  4743.1  257.51  4764.1  258.33  4792.5  257.28  4842.1  257.58  4926.9  255.16
  4934.3  255.63  4955.2  253.62  4976.8  255.47    4991  253.07  4992.2  250.39
  4992.7  249.89  5010.8  250.39  5019.7  255.43  5056.3  260.14  5097.8  260.55
  5103.2  261.56  5146.7  264.09  5229.7  268.56  5259.3   271.6  5274.1  271.63
#Mann= 6 ,-1 , 0
  4190.9     .05       0  4612.4      .1       0  4992.2     .05       0
  5010.8      .1       0  5056.3     .07       0  5146.7      .1       0
Bank Sta=4992.2,5010.8
XS Rating Curve= 0 ,0
Exp/Cntr=0.3,0.1

Type RM Length L Ch R = 1 ,46431   ,467,467,467
BEGIN DESCRIPTION:
MCCOY CREEK 53.0
END DESCRIPTION:
XS GIS Cut Line= 3
        2517725.       13652875.        2517225.       13652425.
      2516624.99     13651974.99
#Sta/Elev= 30
  4332.5   277.2  4336.7  277.19  4410.6  273.74  4424.8  274.11  4465.8  271.56
  4495.1  269.69  4516.7  270.32  4573.5  266.59  4594.5   267.2  4629.6  264.34
  4688.2  261.72  4771.6  259.24  4792.5  257.33  4870.6   255.3  4877.7   254.3
    4963  253.82  4977.2  252.84  4988.8  250.21  4989.3  249.71  5007.4  250.21
  5018.7   252.8  5041.6  253.79  5047.9  255.06  5080.6  254.95  5104.2  254.72
  5191.6  255.36  5404.9  262.05  5465.6  264.63  5529.6  267.57  5755.2  282.69
#Mann= 11 ,-1 , 0
  4332.5     .05       0  4336.7    .035       0  4465.8     .05       0
  4688.2      .1       0  4988.8     .05       0  5007.4      .1       0
  5080.6     .07       0  5104.2     .05       0  5404.9     .07       0
  5465.6     .05       0  5529.6     .07       0
Bank Sta=4988.8,5007.4
XS Rating Curve= 0 ,0
Exp/Cntr=0.3,0.1

Type RM Length L Ch R = 1 ,45964   ,848,848,848
BEGIN DESCRIPTION:
MCCOY CREEK 52.0
END DESCRIPTION:
XS GIS Cut Line= 3
      2517825.02     13652675.04        2517625.       13652225.
        2516525.       13651225.
#Sta/Elev= 30
  4507.9  273.39  4667.3  266.41  4690.6  266.94  4726.8  264.08  4759.6   264.1
  4781.5  261.75  4817.8  263.16  4858.1  261.19    4893  256.15  4908.1   255.8
  4939.5  253.85  4976.7  248.58  4977.2  248.08  4995.3  248.58  4997.7  252.32
  5007.5  253.64  5056.8  252.21  5177.1  255.16  5237.7   253.9  5332.6  253.68
  5367.3  252.86    5497  255.71  5581.2  257.42  5629.9  260.57  5733.1  264.09
  5821.7  266.77  5842.7   269.6  5966.6   276.4  6274.5  298.58    6487  309.22
#Mann= 11 ,-1 , 0
  4507.9     .05       0  4908.1      .1       0  4976.7     .05       0
  4995.3      .1       0  5237.7     .07       0  5332.6     .12       0
  5367.3    .035       0    5497     .12       0  5629.9     .07       0
  5733.1     .12       0  5966.6     .07       0
Bank Sta=4976.7,4995.3
XS Rating Curve= 0 ,0
Exp/Cntr=0.3,0.1

Type RM Length L Ch R = 1 ,45116   ,470,470,470
BEGIN DESCRIPTION:
B19361
END DESCRIPTION:
XS GIS Cut Line= 3
      2517898.82     13652949.21      2517667.38     13651714.87
      2516923.53     13651136.32
#Sta/Elev= 30
  3400.5  282.26  3425.1  283.39  3507.1  279.48    3537  279.84  3598.1   275.8
  3618.4  276.84  3679.5  272.73  3699.8  273.85  3781.2  269.12  3801.6  269.87
  3885.3  266.69  3923.7  263.78  4158.3  258.12  4513.8  253.41    4824  252.91
  4900.1  253.22    4922  250.44  4963.6  249.95  4991.4  247.13  4991.9  246.63
    5010  247.13  5014.1  250.04  5021.5  251.41  5077.6  255.61  5121.1  262.85
  5158.3  266.06  5280.3  274.33  5323.5  277.17  5402.3  282.42  5598.7  297.94
#Mann= 8 ,-1 , 0
  3400.5     .05       0    4824      .1       0  4991.4     .05       0
    5010      .1       0  5158.3    .035       0  5280.3     .07       0
  5323.5    .035       0  5402.3     .07       0
Bank Sta=4991.4,5010
XS Rating Curve= 0 ,0
Exp/Cntr=0.3,0.1

Type RM Length L Ch R = 1 ,44646   ,442,442,442
BEGIN DESCRIPTION:
MCCOY CREEK 51.0
END DESCRIPTION:
XS GIS Cut Line= 3
        2517925.     13652974.99        2517625.       13651175.
      2517275.02     13650975.01
#Sta/Elev= 30
  3175.1  284.39  3215.6  282.36  3246.1  283.08  3324.6  279.02  3347.4  279.65
  3408.3  275.74  3428.5  276.72  3479.2   273.2  3512.2  273.57  3580.6  269.55
    3611  269.74  3742.8  263.68  3773.2  264.19  3811.2  261.53  3834.1  262.59
  3932.9  258.78    4270  254.37  4792.1  251.78  4911.2  251.51  4970.3  246.25
  4970.8  245.75    4989  246.25    5023  250.05  5035.2  253.36  5112.4  260.48
  5233.9  268.69  5264.8   272.2  5299.4  278.96  5375.8  286.61    5403  287.42
#Mann= 6 ,-1 , 0
  3175.1     .05       0  4792.1      .1       0  4970.3     .05       0
    4989      .1       0  5112.4     .12       0  5375.8     .07       0
Bank Sta=4970.3,4989
XS Rating Curve= 0 ,0
Exp/Cntr=0.3,0.1

Type RM Length L Ch R = 1 ,44204   ,471,471,471
BEGIN DESCRIPTION:
MCCOY CREEK 50.0
END DESCRIPTION:
XS GIS Cut Line= 3
      2518524.98     13651574.97        2517975.       13650975.
      2517374.98       13650875.
#Sta/Elev= 30
  4181.8  266.31  4253.4  264.02  4351.6  258.76  4429.3  256.74  4450.9  257.63
  4471.9  256.98  4479.3  255.51  4486.1  255.98  4493.5  254.19  4550.9  254.77
    4557  255.56  4592.1  255.37  4634.7  253.74  4804.9  251.54  4841.6  250.23
  4967.6   250.5  4981.8  249.45  4982.5   244.4    4983   243.9  5002.1   244.4
  5005.8  246.06    5016  247.04  5046.4  246.41  5066.7  249.03  5178.2  252.45
    5296  258.28    5495  269.06    5571  274.45  5576.1  273.95    5604   275.8
#Mann= 8 ,-1 , 0
  4181.8     .05       0  4253.4     .07       0  4550.9     .05       0
  4841.6      .1       0  4982.5     .05       0  5002.1      .1       0
    5296     .07       0    5495     .12       0
Bank Sta=4982.5,5002.1
XS Rating Curve= 0 ,0
Exp/Cntr=0.3,0.1

Type RM Length L Ch R = 1 ,43733   ,428,428,428
BEGIN DESCRIPTION:
MCCOY CREEK 49.0
END DESCRIPTION:
XS GIS Cut Line= 3
      2518825.03     13651125.03        2518225.       13650625.
      2517624.98     13650224.99
#Sta/Elev= 30
  4218.7  271.42    4261  270.07  4324.8  265.88  4339.1  266.32  4410.7  261.56
  4425.1  262.21    4453  259.42    4481  259.32  4538.3  255.97  4559.1  256.15
  4622.9  253.69  4630.7  254.71  4673.7  252.76  4901.9  249.65    4964  249.49
  4971.8  248.04  4978.3  248.37  4982.8  243.91  4983.3  243.41  5002.4  243.91
  5002.8  244.84  5007.3   246.1  5094.4  249.42  5193.6  249.89  5403.9  253.96
  5468.5  254.21  5515.8  256.19  5518.6  256.26  5634.7  261.56  5720.9  265.44
#Mann= 7 ,-1 , 0
  4218.7     .05       0  4901.9      .1       0  4982.8     .05       0
  5002.4      .1       0  5515.8     .07       0  5518.6      .1       0
  5634.7     .12       0
Bank Sta=4982.8,5002.4
XS Rating Curve= 0 ,0
Exp/Cntr=0.3,0.1

Type RM Length L Ch R = 1 ,43305   ,485,485,485
BEGIN DESCRIPTION:
MCCOY CREEK 48.0
END DESCRIPTION:
XS GIS Cut Line= 3
      2518825.01       13650175.        2518425.       13650275.
      2517224.97       13650075.
#Sta/Elev= 30
  4592.8  266.39  4657.2  263.12  4693.3  259.55  4734.5  257.25  4854.1  253.31
  4881.4  252.31  4904.6  249.47  4912.3   246.6  4940.7  245.12  4945.8   246.6
  4953.6   243.1  4963.9  243.54  4972.1  241.86  4972.6  241.36  4991.7  241.86
  5007.7  243.17  5015.3  245.02  5045.7  247.62  5141.2  247.96  5144.1  248.03
  5248.4  247.04  5442.2  250.69  5536.7  254.02  5646.3  258.43  5888.2  271.07
  5958.1  275.85  6039.2  279.22    6100  283.94  6197.7  287.46  6221.7  288.67
#Mann= 10 ,-1 , 0
  4592.8     .05       0  4854.1      .1       0  4972.1     .05       0
  4991.7      .1       0  5141.2     .07       0  5144.1      .1       0
  5442.2     .12       0  5536.7     .07       0  5888.2     .12       0
  6197.7     .07       0
Bank Sta=4972.1,4991.7
XS Rating Curve= 0 ,0
Exp/Cntr=0.3,0.1

Type RM Length L Ch R = 1 ,42820   ,453,453,453
BEGIN DESCRIPTION:
MCCOY CREEK 47.0
END DESCRIPTION:
XS GIS Cut Line= 3
      2518825.02     13649724.99        2518525.       13649825.
      2517424.99       13650025.
#Sta/Elev= 30
  4684.2  264.69  4723.4   262.6    4758  258.86  4800.2  256.08    4926  251.79
  4947.7  250.22  4968.8   246.7  4980.1  240.97  4980.6  240.47  4999.8  240.97
  5000.5  242.43  5010.6  243.02  5027.1  246.31  5051.3  247.14  5091.9  245.65
  5122.4  246.85  5203.7  247.52  5244.4  246.71  5264.7  245.19  5331.1  246.69
  5396.8  246.72    5421  245.93  5508.6  247.12    5646  252.45  5756.4  257.13
  5783.1  259.29  5823.7  264.22  5863.1  267.29  6060.8  276.29  6118.5  280.91
#Mann= 8 ,-1 , 0
  4684.2     .05       0  4723.4     .07       0    4926      .1       0
  4980.1     .05       0  4999.8      .1       0  5331.1     .12       0
    5646     .07       0  6060.8     .12       0
Bank Sta=4980.1,4999.8
XS Rating Curve= 0 ,0
Exp/Cntr=0.3,0.1

Type RM Length L Ch R = 1 ,42367   ,1592,1592,1592
BEGIN DESCRIPTION:
MCCOY CREEK 46.0
END DESCRIPTION:
XS GIS Cut Line= 3
      2518875.01       13649525.        2518375.       13649425.
      2517275.01       13650025.
#Sta/Elev= 30
    4490  265.91  4565.9  261.45  4665.7  255.42  4741.3  251.86  4765.5  251.13
  4867.3  247.77  4918.3  247.58  4959.1  245.42  4979.5  241.92  4979.9  239.39
  4980.4  238.89  4999.6  239.39  4999.9   241.8  5002.8   241.8    5008  244.76
  5022.7  245.89  5148.5  245.26    5282   245.4  5301.6  245.06  5367.7  245.57
  5405.7  242.23  5411.4   244.7  5580.8  247.23  5759.8  254.24  5866.5  261.25
  5906.9  263.58  5994.2  271.98    6103  279.25  6245.8   286.5  6252.9  287.13
#Mann= 13 ,-1 , 0
    4490     .05       0  4565.9     .07       0  4665.7      .1       0
  4741.3     .07       0  4765.5      .1       0  4979.9     .05       0
  4999.6      .1       0  5148.5     .12       0    5282     .07       0
  5301.6     .12       0  5866.5     .07       0    6103     .12       0
  6245.8     .07       0
Bank Sta=4979.9,4999.6
XS Rating Curve= 0 ,0
Exp/Cntr=0.3,0.1

Type RM Length L Ch R = 1 ,40775   ,983,983,983
BEGIN DESCRIPTION:
B19360
END DESCRIPTION:
XS GIS Cut Line= 3
      2519420.06     13648818.73      2517861.42      13648796.3
       2516348.8     13649614.24
#Sta/Elev= 30
    2691  268.46  3046.1  267.69  3126.1  264.19  3299.4   261.1  3435.3  256.56
  3626.2  250.51  3782.7  248.58  3897.9  249.83  3966.2  251.86  4156.2  250.15
  4527.6  243.71  4797.6  242.66  4931.9  241.64  4961.9  239.48    4982  234.37
  4982.5  233.87  5001.8  234.37  5007.4  244.57  5013.1  245.91    5019  247.92
  5095.6  255.94  5243.3  259.89  5308.7  264.28  5330.6  263.83  5434.3  268.96
  5478.1  269.06  5507.6  272.29  5607.3  275.03  5838.7  284.51  5969.4  287.55
#Mann= 11 ,-1 , 0
    2691     .05       0  3435.3     .07       0  3782.7      .1       0
  3897.9     .05       0  4797.6     .07       0    4982     .05       0
  5001.8     .07       0  5013.1      .1       0    5019     .07       0
  5243.3     .05       0  5607.3     .07       0
Bank Sta=4982,5001.8
XS Rating Curve= 0 ,0
Exp/Cntr=0.3,0.1

Type RM Length L Ch R = 1 ,39792   ,651,651,651
BEGIN DESCRIPTION:
B19359
END DESCRIPTION:
XS GIS Cut Line= 3
      2519464.98     13648729.03      2517031.63     13648190.78
       2516404.5     13648750.72
#Sta/Elev= 30
    2825  267.42  3287.2   264.8  4079.8  244.16  4179.9  242.68  4380.2  241.36
  4480.4  240.97  4482.3  240.97  4703.6  240.19  4762.3  240.78  4857.9  239.95
    4881  240.97  4950.2  240.45  4965.5  236.99  4975.7  233.01  4976.1   231.7
  4976.6   231.2  4995.9   231.7    4999  236.35  5057.7  244.28  5108.9  246.66
  5190.8  252.89    5242  254.89  5322.9   255.2  5540.3  258.79  5544.8  258.82
  5688.2  261.56  5810.4  262.04  5831.5  261.83  5996.8  261.54  6157.9  263.42
#Mann= 18 ,-1 , 0
    2825     .05       0  4079.8     .07       0  4179.9     .12       0
  4380.2     .07       0  4480.4     .12       0  4482.3     .07       0
  4703.6      .1       0  4762.3     .07       0    4881     .05       0
  4976.1     .05       0  4995.9     .05       0  5322.9     .07       0
  5540.3     .12       0  5544.8    .035       0  5688.2     .12       0
  5810.4     .07       0  5831.5     .12       0  5996.8     .05       0
Bank Sta=4976.1,4995.9
XS Rating Curve= 0 ,0
Exp/Cntr=0.3,0.1

Type RM Length L Ch R = 1 ,39141   ,1281,1281,1281
BEGIN DESCRIPTION:
B19358
END DESCRIPTION:
XS GIS Cut Line= 3
      2519532.18     13648661.72      2517525.02     13647652.54
      2516438.65     13648638.11
#Sta/Elev= 30
    2956  265.83  3271.7  264.27  3377.7  265.38  3986.6  242.23  4124.4  239.16
  4309.6  238.05  4536.2  238.25  4686.7  238.68  4962.7  239.15    4985  237.37
  5001.1   234.1    5003  229.76  5003.5  229.26  5022.8  229.76  5023.5  231.61
  5035.2  236.91  5044.4  238.83  5079.9  244.34  5239.9  241.47  5303.4  243.67
  5431.2  244.19  5706.9  251.79  5896.6  253.19  6103.4  256.68  6225.3  259.26
  6367.5  260.94  6509.7  261.42  6634.9  261.85  6651.9  261.92  6669.4  261.45
#Mann= 16 ,-1 , 0
    2956     .05       0  3986.6     .12       0  4124.4     .05       0
  4309.6      .1       0  4536.2     .05       0  4686.7      .1       0
    5003     .05       0  5022.8      .1       0  5044.4     .05       0
  5896.6     .07       0  6103.4     .12       0  6225.3    .035       0
  6367.5     .07       0  6509.7     .12       0  6634.9     .07       0
  6651.9     .05       0
Bank Sta=5003,5022.8
XS Rating Curve= 0 ,0
Exp/Cntr=0.3,0.1

Type RM Length L Ch R = 1 ,37860   ,921,921,921
BEGIN DESCRIPTION:
B19357
END DESCRIPTION:
XS GIS Cut Line= 4
        2519678.     13648661.75      2518736.07     13647417.05
      2517782.93     13647327.35      2516459.89     13648549.48
#Sta/Elev= 30
  3686.6  265.93  3879.5  264.86  3914.9  261.64  4035.6  259.26  4443.4  257.38
  4887.1  240.94  4957.3  238.02  4986.5  232.07  4989.3  227.46  4989.8  226.96
  5009.2  227.46  5013.6  231.94  5021.8  234.51  5081.8  236.45    5349  237.13
  5449.5  232.79  5535.5  237.16  5690.5  235.88    6022  242.93  6265.5  239.06
  6576.8  238.35  6838.8  241.36  7022.5  249.09    7275  251.36  7472.8  254.87
  7693.6  258.89  7834.5  261.12  7975.4  260.99  7997.4  260.99    8006  260.75
#Mann= 11 ,-1 , 0
  3686.6     .05       0  4887.1      .1       0  4989.3     .05       0
  5009.2      .1       0  5081.8     .05       0    7275     .07       0
  7472.8     .12       0  7693.6    .035       0  7834.5     .07       0
  7975.4     .12       0  7997.4     .07       0
Bank Sta=4989.3,5009.2
XS Rating Curve= 0 ,0
Exp/Cntr=0.3,0.1

Type RM Length L Ch R = 1 ,36939   ,1234,1234,1234
BEGIN DESCRIPTION:
B19356
END DESCRIPTION:
XS GIS Cut Line= 5
      2520512.61      13648289.8      2519195.82     13646833.96
      2518545.44     13646811.53      2517827.78     13647237.64
      2516515.79     13648448.71
#Sta/Elev= 30
  2916.2  260.63  3065.5  256.25  3338.8  248.91  3382.5  246.55  3399.2  248.53
  3492.3  246.58  3602.6  245.34  3753.9  245.09  3976.9  242.09  4291.4  236.11
  4745.4  235.77  4884.8  235.74  4960.1  235.12  4980.1  230.88  4990.1  225.01
  4990.6  224.51  5010.1  225.01  5020.1  232.38  5030.1   233.7  5136.2  234.22
  5903.8  233.49  6196.1  243.63  6824.7  236.75  7044.2   238.8  7298.8  248.99
  7507.3  250.21  7698.7  253.97    7984  258.94    8125  260.16  8150.1  259.76
#Mann= 17 ,-1 , 0
  2916.2     .05       0  3065.5     .12       0  3338.8     .07       0
  3382.5      .1       0  3492.3     .07       0  3602.6     .05       0
  3753.9     .07       0  3976.9     .05       0  4745.4     .07       0
  4884.8      .1       0  4990.1     .05       0  5010.1      .1       0
  5136.2     .05       0  7507.3     .07       0  7698.7     .12       0
    7984    .035       0    8125     .07       0
Bank Sta=4990.1,5010.1
XS Rating Curve= 0 ,0
Exp/Cntr=0.3,0.1

Type RM Length L Ch R = 1 ,35705   ,877,877,877
BEGIN DESCRIPTION:
B19355
END DESCRIPTION:
XS GIS Cut Line= 4
      2518342.49     13644887.06      2518213.42      13645909.3
      2517883.85     13647114.29      2516594.28     13648325.37
#Sta/Elev= 30
  3331.3  274.84  3748.9  287.61  3841.4  288.64    3934  287.44  4105.3  279.02
  4419.4  257.21  4447.9  253.02  4668.2  238.35  4761.5  234.51  4877.2  232.64
    4917  230.38  4968.9  231.02  4977.6  225.86  4981.7  220.87  4982.6  220.37
  5018.2  220.87  5022.4  228.09  5031.1  230.77  5116.3  229.67  5155.5  228.85
    5311  236.93  5456.1  241.03  5652.9  242.29    6028  235.55  6247.3  235.33
  6494.9  240.01  6671.7  247.88  6853.8   248.9  7038.9  252.04    7380  259.06
#Mann= 8 ,-1 , 0
  3331.3     .07       0  3841.4     .05       0  4877.2      .1       0
  4981.7     .05       0  5018.2      .1       0  5116.3     .05       0
  6853.8     .07       0  7038.9     .12       0
Bank Sta=4981.7,5018.2
XS Rating Curve= 0 ,0
Exp/Cntr=0.3,0.1

Type RM Length L Ch R = 1 ,34828   ,710,710,710
BEGIN DESCRIPTION:
B19354
END DESCRIPTION:
XS GIS Cut Line= 3
      2517569.88     13646262.05      2517244.69     13647271.28
      2516627.95     13648213.21
#Sta/Elev= 30
  4304.1  258.49  4436.3   252.6  4644.8  238.95  4747.4  234.92  4810.2   232.1
  4959.8  228.37  4969.1  227.45  4979.6  222.69  4982.3  217.08  4983.2  216.58
  5018.9  217.08  5042.6  220.42  5050.8  227.38    5056  222.22  5074.2  227.79
  5105.7  225.64  5168.7  229.74  5245.4  229.55  5619.9  233.48  5678.5  235.37
  5777.5  242.76  5799.2  244.24  5970.1  243.41  6046.3  244.62  6067.4  240.67
  6133.8  249.08  6160.8  246.84  6197.7  248.51  6271.9  250.82  6490.3  255.81
#Mann= 11 ,-1 , 0
  4304.1     .05       0  4644.8     .07       0  4747.4     .12       0
  4810.2      .1       0  4982.3     .05       0  5018.9      .1       0
  5245.4     .05       0  5777.5      .1       0  5970.1     .12       0
  6197.7     .07       0  6271.9     .12       0
Bank Sta=4982.3,5018.9
XS Rating Curve= 0 ,0
Exp/Cntr=0.3,0.1

Type RM Length L Ch R = 1 ,34118   ,511,511,511
BEGIN DESCRIPTION:
MCCOY CREEK 42.0
END DESCRIPTION:
XS GIS Cut Line= 3
      2517424.98     13646375.02        2516775.       13647175.
      2516475.01     13647474.99
#Sta/Elev= 30
  3964.2  254.53    3984  253.74  4145.7  245.89  4270.2  240.68    4469   237.2
  4477.1  236.97  4505.1  237.12  4540.3  235.42  4554.6  236.12    4569   234.6
  4582.6   235.4  4589.4  233.77  4653.8  231.42  4802.4   229.6  4839.1  227.18
  4859.9  226.78  4888.7  227.59    4903  226.61  4923.8   227.6  4944.7  226.99
    4967  228.31  4973.4  217.35  4974.3  216.85  5010.1  217.35  5023.2  223.48
  5051.5  233.14  5065.7  236.92  5165.1  240.13  5221.2  243.38  5419.2   250.3
#Mann= 9 ,-1 , 0
  3964.2     .05       0    3984     .07       0  4145.7     .12       0
    4469      .1       0  4477.1     .12       0  4589.4      .1       0
  4973.4     .05       0  5010.1      .1       0  5165.1     .12       0
Bank Sta=4973.4,5010.1
XS Rating Curve= 0 ,0
Exp/Cntr=0.3,0.1

Type RM Length L Ch R = 1 ,33607   ,529,529,529
BEGIN DESCRIPTION:
MCCOY CREEK 41.0
END DESCRIPTION:
XS GIS Cut Line= 3
        2517175.       13646075.        2516425.       13646875.
        2516225.       13647225.
#Sta/Elev= 30
  3897.4  262.25  3988.4  256.81  4028.8  254.51  4088.6  251.64  4095.5  249.73
  4174.7  247.32  4267.7  242.14  4431.1  235.69  4491.6  233.57  4527.3  234.12
  4576.6  231.78  4776.2   229.4  4788.6  228.31  4895.1  229.02  4951.7   222.7
  4965.9  221.81  4972.7  223.33  4980.1  221.79  4983.6  216.41  4984.5  215.91
  5020.3  216.41  5029.3  219.53  5039.3  219.93  5066.7  225.79  5080.2   226.7
  5132.2  235.56  5191.8  238.74  5281.2  244.69  5304.7   244.4  5397.1  248.54
#Mann= 12 ,-1 , 0
  3897.4     .07       0  3988.4     .12       0  4028.8     .07       0
  4174.7     .12       0  4267.7      .1       0  4431.1     .12       0
  4776.2      .1       0  4983.6     .05       0  5020.3      .1       0
  5080.2     .12       0  5191.8     .05       0  5304.7     .12       0
Bank Sta=4983.6,5020.3
XS Rating Curve= 0 ,0
Exp/Cntr=0.3,0.1

Type RM Length L Ch R = 1 ,33078   ,665,665,665
BEGIN DESCRIPTION:
MCCOY CREEK 40.0
END DESCRIPTION:
XS GIS Cut Line= 3
      2516975.01     13645774.99        2516175.       13646425.
        2516075.     13646925.01
#Sta/Elev= 30
  3959.9  266.81  4125.4  256.93  4222.8  250.57  4301.1  247.87  4336.3  244.25
  4379.4  243.02  4414.6   240.1  4449.8  240.04  4472.1   237.2  4503.5  236.33
  4550.4  235.83  4571.2  234.04  4748.6  229.08  4806.1  228.36  4812.5  229.27
    4849  227.98    4870  229.98  4919.6  230.79  4969.1  224.16  4982.5  215.39
  4983.4  214.89  5019.2  215.39  5021.3  221.25  5031.5  224.36  5062.1  224.29
  5133.5  227.02  5276.2   235.4  5304.3  235.93  5347.6  238.93  5500.6  242.57
#Mann= 6 ,-1 , 0
  3959.9     .12       0  4125.4     .07       0  4503.5      .1       0
  4982.5     .05       0  5019.2      .1       0  5304.3     .05       0
Bank Sta=4982.5,5019.2
XS Rating Curve= 0 ,0
Exp/Cntr=0.3,0.1

Type RM Length L Ch R = 1 ,32413   ,561,561,561
BEGIN DESCRIPTION:
B19353
END DESCRIPTION:
XS GIS Cut Line= 3
      2515786.94      13644905.3      2515652.38     13646228.43
      2515999.99     13647125.48
#Sta/Elev= 30
  3876.3  271.28  4230.3   261.6    4329  258.02  4358.5  257.04  4526.5   246.1
  4601.8  241.58  4635.8  238.76  4680.1  237.33  4735.5  230.81    4851  227.16
  4881.2  224.69  4891.2  225.81  4911.3  224.62  4929.8  220.12  4934.9  225.94
  4951.5  220.69  4971.6  221.57  4973.3  214.77  4974.2  214.27  5010.2  214.77
  5029.5  222.75  5092.2  226.63  5454.5  229.64  5534.9  230.34  5577.9  231.24
  5615.1  230.02  5685.2  230.69  5803.7  234.12  6122.5  244.93  6168.3  246.48
#Mann= 11 ,-1 , 0
  3876.3     .07       0  4230.3     .12       0    4329     .07       0
  4526.5     .12       0  4601.8      .1       0  4973.3     .05       0
  5010.2      .1       0  5454.5    .035       0  5534.9      .1       0
  5803.7     .05       0  6122.5     .07       0
Bank Sta=4973.3,5010.2
XS Rating Curve= 0 ,0
Exp/Cntr=0.3,0.1

Type RM Length L Ch R = 1 ,31852   ,1109,1109,1109
BEGIN DESCRIPTION:
MCCOY CREEK 39.0
END DESCRIPTION:
XS GIS Cut Line= 3
      2515495.38     13644961.36       2515080.5      13646116.3
      2514677.43     13646911.25
#Sta/Elev= 30
  4029.2  254.57    4313  242.95  4338.4  244.03    4456  240.27  4640.4  229.05
  4752.7  227.49  4798.1  224.66  4808.7  226.45  4819.4  224.26  4925.6  220.68
  4931.7  225.46    4937  221.56  4957.1  225.56  4962.5  222.47  4968.1  225.13
  4978.8  225.08  4981.4  216.45  4982.4  215.95  5018.6  216.45  5031.9  224.46
  5049.3  225.14  5095.6     224    5259  226.85  5431.6   222.8  5529.2   226.2
  5541.9  227.59  5701.7  237.24  5795.2  242.31  5871.3  246.57  6147.7  253.48
#Mann= 7 ,-1 , 0
  4029.2      .1       0  4981.4     .05       0  5018.6      .1       0
  5529.2    .035       0  5541.9      .1       0  5701.7     .12       0
  5795.2     .05       0
Bank Sta=4981.4,5018.6
XS Rating Curve= 0 ,0
Exp/Cntr=0.3,0.1
