HEC-RAS study MOUND CREEK.prj: MOUND CREEK Base Level Engineering

--- MOUND CREEK.g01 (geometry) --- (continued)

Type RM Length L Ch R = 1 ,57052   ,908,908,908
BEGIN DESCRIPTION:
MOUND CREEK 78.0
END DESCRIPTION:
XS GIS Cut Line= 3
      2394224.96     13603874.98        2395025.       13604225.
      2395474.97       13604175.
#Sta/Elev= 30
  4132.2  397.75  4186.8  395.44  4216.8  392.33  4252.3  386.03  4285.1  384.46
  4328.7  380.29  4373.5  377.09  4482.7  371.58  4525.2  368.99  4589.5  368.29
  4601.6  367.09  4641.7  369.03  4670.6  368.02  4717.4  368.59  4740.8  367.64
    4793  369.11  4938.8   368.8  4996.5  367.77  5002.7  364.65    5008  364.65
  5009.7  362.91  5010.2  362.41  5021.3  362.91  5025.6  367.96  5035.6   373.3
  5045.7  374.81  5121.8  376.06  5146.3  376.84  5317.4  376.61  5458.2  378.54
#Mann= 5 ,-1 , 0
  4132.2     .07       0  4482.7      .1       0  5009.7     .05       0
  5021.3      .1       0  5121.8     .05       0
Bank Sta=5009.7,5021.3
XS Rating Curve= 0 ,0
Exp/Cntr=0.3,0.1

Type RM Length L Ch R = 1 ,56144   ,435,435,435
BEGIN DESCRIPTION:
B19644
END DESCRIPTION:
XS GIS Cut Line= 4
      2394024.25     13604117.72      2394459.54      13604391.8
      2394642.27     13604569.15      2395217.31     13604563.77
#Sta/Elev= 30
  4584.5  390.66  4656.3  388.03    4663  388.96  4668.9  387.72  4684.2  386.71
  4902.7  376.58  4975.4  373.55  4982.1   372.9    4985  371.66  4997.4  366.96
  5003.3   361.6  5012.8  359.82  5013.3  359.32  5024.4  359.82  5024.5   363.7
  5033.9  365.43  5046.3   366.2  5175.8  366.96  5260.5  365.81    5296  366.67
  5317.1  365.92  5331.2  367.02  5426.3  367.21  5486.3  366.33  5526.3  366.77
  5546.5     368  5596.3  371.06  5644.9  372.79  5716.3  375.22  5928.6  373.68
#Mann= 7 ,-1 , 0
  4584.5     .05       0  4902.7     .07       0    4985      .1       0
  5012.8     .05       0  5024.4      .1       0  5546.5     .07       0
  5644.9     .05       0
Bank Sta=5012.8,5024.4
XS Rating Curve= 0 ,0
Exp/Cntr=0.3,0.1

Type RM Length L Ch R = 1 ,55709   ,479,479,479
BEGIN DESCRIPTION:
MOUND CREEK 77.0
END DESCRIPTION:
XS GIS Cut Line= 3
      2394074.98     13604474.99        2394575.       13604675.
      2394975.05     13604624.99
#Sta/Elev= 30
  4461.3  374.25  4559.6  372.54  4583.8  371.56  4608.1  371.45  4644.4  369.58
  4686.2  369.07  4715.8  367.75  4809.1   366.5  4906.9  365.74  4913.7  365.15
  4967.5   364.6  4978.3  363.93    4985   361.2  4990.4  361.71  4991.3  358.54
  4991.8  358.04  5002.4  358.04  5002.9  358.54  5009.9  361.37    5020  364.18
  5030.1  363.91  5037.6  365.21  5042.7  365.21  5050.2  366.04  5140.9  366.82
  5203.9  365.23  5259.9  367.38  5332.4  371.22  5359.4  371.93    5403  373.58
#Mann= 6 ,-1 , 0
  4461.3     .07       0  4809.1      .1       0  4991.3     .05       0
  5002.9      .1       0  5259.9     .07       0  5359.4     .05       0
Bank Sta=4991.3,5002.9
XS Rating Curve= 0 ,0
Exp/Cntr=0.3,0.1

Type RM Length L Ch R = 1 ,55230   ,420,420,420
BEGIN DESCRIPTION:
MOUND CREEK 76.0
END DESCRIPTION:
XS GIS Cut Line= 3
      2393775.02     13604775.01        2394575.       13605125.
      2395025.02     13604724.98
#Sta/Elev= 30
  4122.4  381.46  4183.6  377.43  4198.8  377.06  4220.6  374.98  4264.7   372.9
  4282.6     373  4433.8  368.57  4685.1   365.8  4702.5  365.76  4913.3  363.84
  4973.8  363.24  4986.6  362.18  4992.9  360.62  4998.9  360.62  5002.7  359.31
  5009.4  363.24  5017.8  357.19  5018.3  356.69  5029.5  357.19  5031.1  360.14
  5045.3  363.37  5066.3  364.14    5116  364.74  5250.2  364.12  5292.9  364.92
  5330.8  364.36  5397.3  366.54  5465.9  368.72  5555.4  373.03  5597.7  374.19
#Mann= 9 ,-1 , 0
  4122.4     .07       0  4685.1      .1       0  4702.5     .07       0
  4913.3      .1       0  5017.8     .05       0  5029.5      .1       0
  5330.8     .05       0  5397.3     .07       0  5465.9     .05       0
Bank Sta=5017.8,5029.5
XS Rating Curve= 0 ,0
Exp/Cntr=0.3,0.1

Type RM Length L Ch R = 1 ,54810   ,404,404,404
BEGIN DESCRIPTION:
B19643
END DESCRIPTION:
XS GIS Cut Line= 3
      2393594.24     13605746.13      2394862.62     13605439.78
      2395330.11     13605316.19
#Sta/Elev= 30
  3755.6  375.05  3901.6  372.94  3986.7  371.25  4185.9  366.93  4294.7  362.92
  4311.9  364.89  4394.2  363.83  4527.9  361.54  4545.9  359.61    4551  361.28
  4558.8   361.4    4649  361.08  4692.5  361.49  4754.3  359.64  4774.8  361.89
  4816.6  362.55  4990.9   362.9  5008.3  361.77  5011.5  361.38  5016.1  356.55
  5016.6  356.05  5027.8  356.55    5032  361.27  5042.3  362.21  5073.3  363.06
  5104.3  361.93  5210.7  365.77  5313.2  368.69  5450.8  372.08    5544   371.9
#Mann= 11 ,-1 , 0
  3755.6     .05       0  3901.6     .07       0  3986.7     .05       0
  4185.9     .07       0    4649      .1       0  4816.6     .12       0
  5008.3      .1       0  5016.1     .05       0  5027.8      .1       0
  5210.7     .07       0  5313.2     .05       0
Bank Sta=5016.1,5027.8
XS Rating Curve= 0 ,0
Exp/Cntr=0.3,0.1

Type RM Length L Ch R = 1 ,54406   ,399,399,399
BEGIN DESCRIPTION:
B19642
END DESCRIPTION:
XS GIS Cut Line= 3
      2393787.78     13606127.69      2395104.46       13605730.
      2395330.07     13605466.79
#Sta/Elev= 30
  3684.2  377.62  3733.5  377.03  3879.1  370.41  3983.2  367.17  3994.7  367.93
  4013.2  366.21  4198.4  362.21  4366.7  361.46  4391.6  360.47  4412.5  356.33
  4437.9  359.42  4476.4  358.66  4607.9  359.73  4684.3  361.73    4705  361.52
  4725.9  359.11  4854.3  361.41  4976.6  361.25  4986.2  360.85  4991.4  359.28
  4991.6  356.05  4992.1  355.55  5003.4  356.05    5008  358.78  5029.6  364.38
  5073.2  365.92  5137.8  367.73  5203.8  369.06  5360.2  371.51  5406.3  372.04
#Mann= 10 ,-1 , 0
  3684.2     .07       0  4013.2     .12       0  4198.4     .07       0
  4476.4      .1       0  4991.6     .05       0  5003.4      .1       0
  5073.2     .07       0  5137.8      .1       0  5203.8    .035       0
  5360.2     .07       0
Bank Sta=4991.6,5003.4
XS Rating Curve= 0 ,0
Exp/Cntr=0.3,0.1

Type RM Length L Ch R = 1 ,54007   ,568,568,568
BEGIN DESCRIPTION:
MOUND CREEK 75.0
END DESCRIPTION:
XS GIS Cut Line= 3
       2393922.1     13606369.54       2395346.3     13606030.96
      2396231.52     13606122.16
#Sta/Elev= 30
  3718.1  374.39  4070.6  363.55  4422.4  360.69  4495.2  360.06  4641.5  357.23
  4669.6  357.54  4687.3  354.94  4706.6  358.76  4718.1  359.22  4893.7  359.25
  4964.8  358.73  4985.4  353.85  4995.6  358.55  5012.1  359.69  5118.3  361.49
  5210.8  362.27  5323.8  360.08  5381.7  358.89  5391.8  356.29    5396  352.84
  5396.5  352.34  5407.8  352.84  5411.9  356.39    5422  357.14  5565.3  357.93
    5613  361.86  5654.6  362.35  5824.1  370.34  5951.5  373.29  6071.9  378.94
#Mann= 10 ,-1 , 0
  3718.1     .07       0  4422.4      .1       0  4495.2     .07       0
  4641.5      .1       0  4893.7     .12       0  5118.3     .07       0
  5323.8      .1       0    5396     .05       0  5407.8      .1       0
  5654.6     .07       0
Bank Sta=5396,5407.8
XS Rating Curve= 0 ,0
Exp/Cntr=0.3,0.1

Type RM Length L Ch R = 1 ,53439   ,1115,1115,1115
BEGIN DESCRIPTION:
MOUND CREEK 74.0
END DESCRIPTION:
XS GIS Cut Line= 3
      2394104.81     13606606.01      2395281.81     13606391.04
      2396286.81     13606176.06
#Sta/Elev= 30
  4115.5  373.81  4125.9  371.86  4208.4  368.34  4636.4  360.62  4959.4  357.91
  4984.3  356.48  4989.9  353.69  5000.1  352.56  5010.2  353.25  5020.4  356.72
  5030.6  357.77  5172.9   358.8  5213.6  357.42  5284.7   357.4  5461.9  359.14
  5489.1  355.64  5506.3  355.28  5511.4  351.27  5523.8  349.23  5524.3  348.73
  5536.2  349.23  5550.4  349.41  5555.8  354.43  5581.1  357.49  5666.5   360.2
  5743.4  368.01  5765.2  368.71  5969.7  370.43  6272.2  380.87  6339.7  381.81
#Mann= 5 ,-1 , 0
  4115.5     .07       0  4636.4      .1       0  5523.8     .05       0
  5536.2      .1       0  5666.5     .07       0
Bank Sta=5523.8,5536.2
XS Rating Curve= 0 ,0
Exp/Cntr=0.3,0.1

Type RM Length L Ch R = 1 ,52324   ,702,702,702
BEGIN DESCRIPTION:
B19641
END DESCRIPTION:
XS GIS Cut Line= 4
      2394146.73     13606783.36      2395232.37     13606794.11
      2395587.07      13606460.9      2396085.89     13606219.54
#Sta/Elev= 30
  3336.7   372.9    3435  371.25    3615  363.13  3767.9  360.95  3836.4  359.82
  4008.7   358.3    4045  357.07    4075  354.09    4085  356.89    4115  355.38
    4125  357.37    4145  355.86    4155  357.74  4253.1  358.26  4550.8  357.08
  4564.9   355.6  4649.9   355.7  4692.4  353.34  4706.6  355.03  4770.1  355.61
  4962.4  354.54  5007.6   352.3  5017.8  348.26  5018.3  347.76  5031.5  348.26
  5035.9  355.15  5040.1  361.73  5047.2  368.77  5256.1  369.77  5463.2  375.54
#Mann= 7 ,-1 , 0
  3336.7     .07       0  3767.9      .1       0  3836.4     .07       0
  4253.1      .1       0  5017.8     .05       0  5031.5      .1       0
  5035.9     .07       0
Bank Sta=5017.8,5031.5
XS Rating Curve= 0 ,0
Exp/Cntr=0.3,0.1

Type RM Length L Ch R = 1 ,51622   ,431,431,431
BEGIN DESCRIPTION:
MOUND CREEK 73.0
END DESCRIPTION:
XS GIS Cut Line= 3
      2394175.01       13606825.        2395375.       13606825.
      2396183.59      13607272.4
#Sta/Elev= 30
  3800.7  372.68  3930.7  369.69  4020.7  364.16  4070.7  364.62  4178.8  361.77
  4197.4  361.76  4500.7   357.6  4520.7   353.4  4550.7   354.7  4560.7  356.52
  4570.7  354.92  4610.7  357.65    4725  358.31  4830.7  358.62  4880.7  356.76
  4950.7  356.52  4970.7  354.86  4983.3  344.59  4983.8  344.09    4998  344.59
  4998.2  346.18  5003.5  346.18  5014.4  353.03  5103.5  353.84  5205.6  358.26
  5377.5  362.26  5442.7  364.49  5457.8  366.39  5654.6  372.96  5924.8  379.36
#Mann= 7 ,-1 , 0
  3800.7     .07       0  4178.8      .1       0  4197.4     .07       0
    4725      .1       0  4983.3     .05       0    4998      .1       0
  5205.6     .07       0
Bank Sta=4983.3,4998
XS Rating Curve= 0 ,0
Exp/Cntr=0.3,0.1

Type RM Length L Ch R = 1 ,51191   ,454,454,454
BEGIN DESCRIPTION:
MOUND CREEK 72.0
END DESCRIPTION:
XS GIS Cut Line= 3
      2394474.97       13607075.        2395175.       13607175.
      2395575.03     13607675.04
#Sta/Elev= 30
  4303.7   364.7  4453.9  361.85  4798.7  355.63  4808.8  353.44    4829  351.26
  4857.2  351.87    4930  353.53  4940.1  352.32  4950.2  349.41  4960.3  349.02
  4970.4  345.87  4993.4  344.79  4993.9  344.29  5008.1  344.79  5008.3  346.66
    5014  346.66    5018  345.04  5032.4  346.44  5038.9   353.4  5046.9  354.09
  5074.9  354.17  5131.7  356.43  5146.1  355.76  5205.7  356.63  5250.8   357.7
  5343.2  359.23  5416.6   362.1  5565.5  371.05  5629.5  376.56  5651.2  377.28
#Mann= 8 ,-1 , 0
  4303.7     .05       0  4453.9     .07       0  4857.2      .1       0
  4993.4     .05       0  5008.1      .1       0  5205.7     .07       0
  5250.8      .1       0  5343.2     .07       0
Bank Sta=4993.4,5008.1
XS Rating Curve= 0 ,0
Exp/Cntr=0.3,0.1

Type RM Length L Ch R = 1 ,50737   ,454,454,454
BEGIN DESCRIPTION:
MOUND CREEK 71.0
END DESCRIPTION:
XS GIS Cut Line= 3
        2394525.       13607475.        2395025.       13607525.
      2395574.97     13607724.99
#Sta/Elev= 30
  4497.4  364.57  4597.9  361.34    4618  361.57  4678.3  359.03  4839.1  355.74
  4869.2  352.85  4905.2  352.14  4952.2  353.79  4959.7  353.27  4969.7  352.17
  4989.8  348.01  4989.9  343.63  4990.4  343.13  5004.8  343.63  5009.9  348.89
  5021.2  351.78  5045.8   350.9  5053.1  349.93    5107  354.72  5193.4  354.87
  5265.9  356.54  5312.9  358.67  5329.8  359.67  5335.7  361.18  5366.3  363.76
  5372.3  365.46    5383  366.75  5483.4   372.3  5508.7  376.18  5585.1  378.39
#Mann= 5 ,-1 , 0
  4497.4     .07       0  4905.2      .1       0  4989.9     .05       0
  5004.8      .1       0  5312.9     .07       0
Bank Sta=4989.9,5004.8
XS Rating Curve= 0 ,0
Exp/Cntr=0.3,0.1

Type RM Length L Ch R = 1 ,50283   ,467,467,467
BEGIN DESCRIPTION:
MOUND CREEK 70.0
END DESCRIPTION:
XS GIS Cut Line= 3
        2394575.       13608075.        2394825.       13607875.
      2395424.96       13607925.
#Sta/Elev= 30
  4680.4  363.66  4751.6   362.7  4794.9  360.84  4879.7  358.64  4914.9  358.43
  4929.3   357.4  4936.5  353.69  4943.7  348.48  4950.1  348.31  4957.1  343.37
  4957.6  342.87  4971.5  342.87    4972  343.37    4976  344.06    4987   345.6
  5050.7  348.26  5058.3  348.73  5063.3  349.82  5090.9  349.39    5141  351.23
  5201.3  352.39  5291.6  352.48  5310.7  353.23  5351.8  353.98  5432.1  358.12
  5492.3  362.96  5544.9  368.66  5552.5  370.28  5572.5  372.72  5602.6  373.63
#Mann= 5 ,-1 , 0
  4680.4     .07       0  4957.1     .05       0    4972     .07       0
    4976      .1       0  5310.7     .07       0
Bank Sta=4957.1,4972
XS Rating Curve= 0 ,0
Exp/Cntr=0.3,0.1

Type RM Length L Ch R = 1 ,49816   ,894,894,894
BEGIN DESCRIPTION:
MOUND CREEK 69.0
END DESCRIPTION:
XS GIS Cut Line= 3
      2394624.96     13608274.99        2394875.       13608325.
      2395474.99       13607975.
#Sta/Elev= 30
  4745.9  362.72  4807.1  361.61  4909.1  357.95  4949.9  355.63  4969.4  353.23
  4998.3  349.12  5003.8  349.12  5014.5  342.53  5016.6  342.26  5017.1  341.76
  5031.5  342.26    5036  349.68    5046  350.11  5147.7  348.75  5278.7  349.07
  5308.1  348.28  5388.3  351.67    5404  353.48  5409.8   352.8  5419.1  353.27
  5452.8  356.86  5468.5  359.24  5475.5  361.52    5495  362.62  5527.2  363.59
  5542.9  365.46  5548.7  365.12  5570.2  366.61  5644.7   373.8  5695.5  375.89
#Mann= 6 ,-1 , 0
  4745.9     .07       0  4969.4      .1       0  5016.6     .05       0
  5031.5      .1       0  5419.1     .12       0    5495     .07       0
Bank Sta=5016.6,5031.5
XS Rating Curve= 0 ,0
Exp/Cntr=0.3,0.1

Type RM Length L Ch R = 1 ,48922   ,183,183,183
BEGIN DESCRIPTION:
MOUND CREEK 68.0
END DESCRIPTION:
XS GIS Cut Line= 3
      2394674.96     13608424.98        2395225.       13608675.
      2395524.96     13608475.03
#Sta/Elev= 30
  4403.2  359.99  4435.1  359.11  4440.6  359.81  4458.2  358.23  4492.2  357.72
  4509.8  356.53  4653.7  352.02  4753.1  350.44  4923.9  349.21  4930.5  348.21
    4934   339.9  4934.5   339.4    4949   339.9  4963.5   340.5    4970  345.55
  4975.5  340.79  4985.4  345.28  4993.1  345.75  4998.6  343.47  5004.6   345.8
  5010.4   345.8  5020.9  347.28    5057  346.98    5108  348.35  5115.6  348.85
  5138.1  352.78  5151.6  353.81  5237.2  356.25  5265.7  358.06  5367.9  365.04
#Mann= 5 ,-1 , 0
  4403.2     .07       0  4753.1      .1       0    4934     .05       0
    4949      .1       0  5265.7     .07       0
Bank Sta=4934,4949
XS Rating Curve= 0 ,0
Exp/Cntr=0.3,0.1

Type RM Length L Ch R = 1 ,48739   ,285,285,285
BEGIN DESCRIPTION:
B19640
END DESCRIPTION:
XS GIS Cut Line= 3
      2394420.86     13608562.26      2395103.39     13608820.22
      2396065.43     13608814.84
#Sta/Elev= 30
  4056.5  361.51    4138  359.95    4193  356.15  4199.9  358.04  4327.9  357.41
  4478.8  351.63  4648.9     349  4759.2  349.95  4788.5   348.4  4957.8  346.08
  4970.2  339.87  4970.7  339.37  4985.3  339.87  4997.8  346.73  5027.8  346.18
  5047.8  350.12  5067.8  349.79  5077.8  347.85  5087.8  342.97  5097.8  347.85
  5107.8  349.08  5227.8  351.85  5307.8  348.25  5327.8  350.44  5347.8  354.99
  5377.8  356.15  5407.9  354.51  5497.8  361.96  5617.8  368.78  5748.2  372.35
#Mann= 6 ,-1 , 0
  4056.5     .07       0  4648.9     .12       0  4788.5      .1       0
  4970.2     .05       0  4985.3      .1       0  5407.9     .07       0
Bank Sta=4970.2,4985.3
XS Rating Curve= 0 ,0
Exp/Cntr=0.3,0.1

Type RM Length L Ch R = 1 ,48454   ,909,909,909
BEGIN DESCRIPTION:
B19639
END DESCRIPTION:
XS GIS Cut Line= 3
       2394361.7     13608734.22      2395194.75     13609072.81
       2395947.1     13609067.44
#Sta/Elev= 30
  3877.1  360.47  4025.8  359.38  4139.7  355.77  4181.1  353.52  4247.7  351.27
  4264.1  351.59  4341.7  350.51  4347.1  349.68  4472.1  348.38    4584  348.69
  4609.4   348.6  4633.5  344.39  4647.1  344.04  4679.5  344.64    4701  346.31
    4779  345.72  4896.6  346.91  4946.6  346.49  4956.6  345.85    4969  341.22
  4969.5  340.72  4984.1  341.22  4996.6   344.7  5006.6   346.5  5056.6  352.39
  5107.3  354.08  5236.6  355.77  5346.6  358.33  5496.6  366.36  5528.7  369.16
#Mann= 6 ,-1 , 0
  3877.1     .07       0  4472.1     .12       0    4584      .1       0
    4969     .05       0  4984.1      .1       0  5107.3     .07       0
Bank Sta=4969,4984.1
XS Rating Curve= 0 ,0
Exp/Cntr=0.3,0.1

Type RM Length L Ch R = 1 ,47545   ,334,334,334
BEGIN DESCRIPTION:
B19638
END DESCRIPTION:
XS GIS Cut Line= 4
      2394216.62     13609196.42      2395033.52      13609303.9
      2395221.62     13609357.65      2395940.89     13609261.03
#Sta/Elev= 30
  4235.1  364.06    4468  355.88  4636.9  351.65  4643.9  350.87  4648.9  351.46
  4727.7  350.84    4768  346.57  4796.2  346.54  4828.6  342.51  4848.7  346.11
  4866.6  346.57  4948.5  345.98  4959.7  345.01  4972.2  337.82  4972.7  337.32
  4987.4  337.82  4989.9  343.38    5000  344.05    5071  343.86  5117.7  347.04
    5123   348.4  5143.8  349.39  5220.6  348.71  5278.3  348.22  5393.6  350.33
    5470  352.38  5681.9  353.26  5760.2  354.47  5873.6  357.66  5980.4  364.51
#Mann= 7 ,-1 , 0
  4235.1     .07       0    4468     .12       0  4866.6      .1       0
  4972.2     .05       0  4987.4      .1       0  5220.6     .12       0
  5393.6     .07       0
Bank Sta=4972.2,4987.4
XS Rating Curve= 0 ,0
Exp/Cntr=0.3,0.1

Type RM Length L Ch R = 1 ,47211   ,856,856,856
BEGIN DESCRIPTION:
B19637
END DESCRIPTION:
XS GIS Cut Line= 3
      2394270.36     13609862.83      2394705.69     13609669.36
      2395881.38     13609368.72
#Sta/Elev= 30
  4297.7     367  4390.3  365.01  4456.9  361.68  4575.7  359.35  4645.1  357.56
  4729.6  355.39  4770.2  352.68  4856.7   349.1  4945.4  347.65  4968.8  347.64
  4979.8  345.99  4990.1  342.59  5000.5  340.81  5007.1  336.99  5007.6  336.49
  5022.5  336.99  5031.4  343.18  5041.7  344.13  5062.4  343.32    5083  344.88
  5172.9  344.23  5196.6  345.24  5248.2   342.6  5268.8  345.63  5295.4  347.24
    5396  349.81  5516.5  351.98  5846.8  353.09  5929.4  355.47  5987.6  358.61
#Mann= 7 ,-1 , 0
  4297.7     .12       0  4575.7     .07       0  4645.1     .12       0
  4945.4      .1       0  5007.1     .05       0  5022.5      .1       0
    5396     .07       0
Bank Sta=5007.1,5022.5
XS Rating Curve= 0 ,0
Exp/Cntr=0.3,0.1

Type RM Length L Ch R = 1 ,46355   ,803,803,803
BEGIN DESCRIPTION:
B19636
END DESCRIPTION:
XS GIS Cut Line= 3
      2394313.41     13610083.17      2395060.39      13609911.2
      2396049.22     13609588.75
#Sta/Elev= 30
  3835.4  368.78  3960.2  365.49  4165.4  357.45  4257.8  352.79  4309.1  354.75
  4385.2  352.85  4483.5  347.67  4503.3  345.47  4565.9  344.53  4640.8  344.84
  4722.5  347.27  4795.1  343.68  4832.2  343.95  4858.9  340.97  4864.2  341.96
  4869.7  340.21  4896.1  342.22  4974.9  342.76  4985.4  340.84  4989.3  335.29
  4989.8  334.79  5004.7  335.29  5006.5  338.31  5028.9  344.49    5038  348.98
  5101.1   349.7  5143.2  347.95  5165.3  349.42  5480.9  352.99    5642  358.25
#Mann= 7 ,-1 , 0
  3835.4     .12       0  4165.4     .07       0  4503.3     .12       0
  4565.9      .1       0  4989.3     .05       0  5004.7      .1       0
  5165.3     .07       0
Bank Sta=4989.3,5004.7
XS Rating Curve= 0 ,0
Exp/Cntr=0.3,0.1

Type RM Length L Ch R = 1 ,45552   ,445,445,445
BEGIN DESCRIPTION:
B19635
END DESCRIPTION:
XS GIS Cut Line= 3
      2394426.24     13610319.64      2395232.37     13610228.28
      2396311.29     13609900.85
#Sta/Elev= 30
  4347.1  366.26  4506.9  361.78  4537.1  359.92  4611.4  357.58    4688  353.34
  4728.3  349.69  4758.5  352.22  4900.1  348.26  4929.6  346.51  4965.2  339.61
  4970.2  339.63  4972.1  333.93  4972.6  333.43  4987.6  333.93  4989.9   335.8
    5000  339.65  5030.2  340.94  5070.5  339.95  5090.6  342.88  5144.5  345.21
  5202.9  347.02  5301.9  345.13    5433  344.49  5706.6  348.45  5788.2  347.47
  5805.3  348.91  5810.5  348.39  5850.9   350.2  6101.7  354.53  6285.9  359.96
#Mann= 5 ,-1 , 0
  4347.1     .12       0  4900.1      .1       0  4972.1     .05       0
  4987.6      .1       0  5301.9     .07       0
Bank Sta=4972.1,4987.6
XS Rating Curve= 0 ,0
Exp/Cntr=0.3,0.1

Type RM Length L Ch R = 1 ,45107   ,740,740,740
BEGIN DESCRIPTION:
B19634
END DESCRIPTION:
XS GIS Cut Line= 4
      2394523.01     13610448.64       2395162.5     13610599.11
      2395511.83     13610529.24      2396667.31     13610222.91
#Sta/Elev= 30
  4184.7   363.2  4293.3  360.89  4535.4  351.88  4588.1  352.06  4625.3  348.39
  4673.4  349.21  4731.2  344.12  4751.8  345.95  4772.3  339.38  4831.7   338.2
  4854.4  338.15    4884   345.6  4905.4  342.18    4922  343.31  4956.4  343.88
    4986  340.91  4999.5   333.4    5000   332.9  5015.2   333.4  5027.8  338.63
    5037  339.67  5270.7  338.63  5351.1   342.3  5377.1  341.58  5408.1  337.35
  5449.5  338.21  5501.2  343.99  5521.9   342.7  5595.2   345.7  6393.3  365.91
#Mann= 8 ,-1 , 0
  4184.7     .12       0  4293.3     .07       0  4673.4      .1       0
  4831.7     .12       0    4922      .1       0  4999.5     .05       0
  5015.2      .1       0  5595.2     .07       0
Bank Sta=4999.5,5015.2
XS Rating Curve= 0 ,0
Exp/Cntr=0.3,0.1

Type RM Length L Ch R = 1 ,44367   ,535,535,535
BEGIN DESCRIPTION:
B19633
END DESCRIPTION:
XS GIS Cut Line= 4
      2394716.45     13610900.07      2395699.93     13610857.08
      2396070.76      13610685.1      2396737.13     13610287.42
#Sta/Elev= 30
  3712.4  354.43  3845.1  352.12  3899.3  350.94  4240.9  346.88  4505.2  342.53
  4767.7  340.45  4899.6  338.67  4905.1  339.47  4922.5  339.15    4928  337.85
  4950.9   337.6  4956.4  334.51  4965.9  331.91  4966.4  331.41  4981.7  331.91
  5002.2  336.87  5019.6  337.92  5025.1  340.58  5042.5  341.75    5048  344.55
  5070.2  345.51  5088.2   344.8  5099.3  346.02  5110.6  344.68  5115.9  346.02
  5123.9  346.08  5450.7  351.36  5530.5  354.01    5583  354.63  5881.6  365.02
#Mann= 9 ,-1 , 0
  3712.4    .035       0  3845.1     .05       0  3899.3     .07       0
  4240.9     .05       0  4505.2     .07       0  4767.7      .1       0
  4965.9     .05       0  4981.7      .1       0  5123.9     .07       0
Bank Sta=4965.9,4981.7
XS Rating Curve= 0 ,0
Exp/Cntr=0.3,0.1

Type RM Length L Ch R = 1 ,43832   ,466,466,466
BEGIN DESCRIPTION:
MOUND CREEK 63.0
END DESCRIPTION:
XS GIS Cut Line= 3
      2394974.95     13610924.99        2396075.       13611125.
        2396425.       13611375.
#Sta/Elev= 30
  3890.4  350.01    3892  350.01  4100.5  346.83  4328.2  345.56  4753.3   340.4
  4805.2  340.16    4870  336.69  4923.4  336.88  4928.4  331.63  4947.5  329.55
  4967.8   337.4  5011.6  337.19  5013.3  328.98  5013.8  328.48  5030.6  328.98
  5036.7  335.07  5045.3  338.69  5072.4  337.48  5101.9  339.07  5140.6  338.44
  5143.7  338.26  5152.3  333.39  5158.4   333.9    5167  338.26  5180.5  336.44
    5194   337.3  5244.4   343.4  5301.1  347.55  5410.3  355.36  5438.6  356.16
#Mann= 9 ,-1 , 0
  3890.4     .05       0    3892     .07       0  4100.5     .05       0
  4328.2     .07       0  4753.3      .1       0  5013.3     .05       0
  5030.6      .1       0  5140.6     .12       0  5301.1     .07       0
Bank Sta=5013.3,5030.6
XS Rating Curve= 0 ,0
Exp/Cntr=0.3,0.1

Type RM Length L Ch R = 1 ,43366   ,453,453,453
BEGIN DESCRIPTION:
MOUND CREEK 62.0
END DESCRIPTION:
XS GIS Cut Line= 3
      2394574.98       13611425.        2395775.       13611425.
        2396375.       13611475.
#Sta/Elev= 30
  3800.5  362.13  3903.9  357.53  3980.5  353.28  4042.3  351.18  4100.5  348.76
  4269.9  345.31  4325.4  344.61  4540.5  341.99  4910.5  341.18  4940.5  341.89
  4970.5  341.04  4980.5  332.35  4981.9  329.78  4982.4  329.28  4999.2  329.78
  5000.5  331.77    5003  331.77  5010.6  336.29  5020.6  337.74  5070.8   336.5
  5110.9  337.32    5131  336.44  5191.2  337.03  5231.3     336  5271.5  339.11
  5299.3  340.34  5304.1  339.82  5351.7  342.61  5492.2  347.52  5602.6  353.79
#Mann= 8 ,-1 , 0
  3800.5     .07       0  3903.9     .05       0  4042.3     .07       0
  4269.9     .05       0  4325.4     .07       0  4981.9     .05       0
  4999.2     .07       0  5299.3     .07       0
Bank Sta=4981.9,4999.2
XS Rating Curve= 0 ,0
Exp/Cntr=0.3,0.1

Type RM Length L Ch R = 1 ,42913   ,468,468,468
BEGIN DESCRIPTION:
MOUND CREEK 61.0
END DESCRIPTION:
XS GIS Cut Line= 3
      2394824.98       13611625.        2395925.       13611825.
      2396225.04       13611825.
#Sta/Elev= 30
  3885.4  356.18  3917.2  355.51  3965.5  352.73  3970.5  353.12  4058.2  347.74
  4300.9   340.9  4342.8  338.06  4393.6  340.51  4454.6  339.02  4495.3  340.92
  4524.5  341.32  4617.5  339.93  4636.3  340.27  4678.2  335.05  4688.4  334.69
  4800.2  336.02    4851  335.34    4912   336.2  4948.9  334.88  4962.8  332.69
  4971.7  328.32  4974.4  327.75  4974.9  327.25  4991.8  327.75  4993.3  332.76
  5000.9  336.98  5043.5  338.77  5093.5   342.7  5143.5  344.82  5303.5  349.18
#Mann= 5 ,-1 , 0
  3885.4     .07       0  4617.5      .1       0  4948.9     .07       0
  4974.4     .05       0  4991.8     .07       0
Bank Sta=4974.4,4991.8
XS Rating Curve= 0 ,0
Exp/Cntr=0.3,0.1

Type RM Length L Ch R = 1 ,42445   ,433,433,433
BEGIN DESCRIPTION:
MOUND CREEK 60.0
END DESCRIPTION:
XS GIS Cut Line= 3
      2394924.97     13611774.99        2395525.       13611925.
      2396125.03     13612075.01
#Sta/Elev= 30
  4377.8  354.98  4560.8  344.17  4666.4  339.72    4718  339.67  4790.1  338.56
  4808.2  337.61  4821.1  338.84  4878.1  337.87  4890.6  336.57  4895.8  337.21
  4903.5  335.89  4924.1  334.76  4944.8  335.11  4973.1  334.11  4978.8  332.48
    4985   326.2  4985.5   325.7  5002.5   326.2  5006.6  328.87  5019.5  334.35
  5079.5  335.64    5138  336.52  5161.2  335.85  5220.5  338.39  5225.6  337.74
  5261.7  339.39  5266.9  338.36    5299  339.42  5555.5  344.68  5614.8  346.99
#Mann= 7 ,-1 , 0
  4377.8     .07       0  4878.1      .1       0  4978.8     .07       0
    4985     .05       0  5002.5     .07       0  5079.5      .1       0
    5299     .07       0
Bank Sta=4985,5002.5
XS Rating Curve= 0 ,0
Exp/Cntr=0.3,0.1

Type RM Length L Ch R = 1 ,42012   ,481,481,481
BEGIN DESCRIPTION:
MOUND CREEK 59.0
END DESCRIPTION:
XS GIS Cut Line= 3
      2394925.03     13611825.02        2395525.       13612325.
      2395925.01       13612475.
#Sta/Elev= 30
  4214.8  354.77  4250.6  352.91  4271.4  350.11  4335.2  344.92  4357.3  345.18
    4399  340.63    4563  336.52  4683.4  336.44  4711.4     332    4783  332.25
  4811.6  330.62  4834.3  331.88  4861.1  331.82  4901.1  334.44  4939.2   334.2
  4945.7  335.22  4953.5   333.9  4998.5  332.24  5005.6  330.12  5008.4  324.47
  5008.9  323.97  5025.9  324.47  5027.8  329.54  5035.8  333.56  5041.2  333.16
  5059.9  336.49    5091  338.63  5134.6  340.38  5252.1  341.53    5423   345.3
#Mann= 5 ,-1 , 0
  4214.8     .07       0  4834.3      .1       0  4901.1     .07       0
  5008.4     .05       0  5025.9     .07       0
Bank Sta=5008.4,5025.9
XS Rating Curve= 0 ,0
Exp/Cntr=0.3,0.1

Type RM Length L Ch R = 1 ,41531   ,491,491,491
BEGIN DESCRIPTION:
MOUND CREEK 58.0
END DESCRIPTION:
XS GIS Cut Line= 3
      2394875.01     13611925.02        2395175.       13612525.
      2395774.99     13612824.99
#Sta/Elev= 30
  4323.5  350.44  4331.9  348.56  4337.4  349.04  4354.2  344.53  4368.2   342.5
  4421.3  339.57  4622.5  335.21    4851  334.35  4896.5  334.59  4918.8  331.82
  4971.9  332.41  4997.1   330.9  5002.7  329.89  5007.9  322.75  5008.4  322.25
  5025.5  322.75  5030.6  327.14    5039  330.44    5053  333.79  5075.4  334.97
  5102.8  333.66  5120.1  334.15  5136.8  337.35  5150.8  338.24  5191.1  338.81
  5248.6  338.24    5299  339.18  5382.8  337.11  5500.2  336.33  5665.1  344.11
#Mann= 6 ,-1 , 0
  4323.5     .07       0    4851      .1       0  5007.9     .05       0
  5025.5      .1       0  5102.8     .12       0  5191.1     .07       0
Bank Sta=5007.9,5025.5
XS Rating Curve= 0 ,0
Exp/Cntr=0.3,0.1

Type RM Length L Ch R = 1 ,41040   ,456,456,456
BEGIN DESCRIPTION:
MOUND CREEK 57.0
END DESCRIPTION:
XS GIS Cut Line= 3
      2394224.98     13612174.98        2394725.       13612625.
      2395925.03     13613825.03
#Sta/Elev= 30
  4323.6  363.45  4359.1  362.59  4592.7  342.34  4628.2  334.53  4649.1  332.32
  4720.1   331.6  4797.9  334.24  4946.6  332.82  4960.8     332  4968.3   326.7
  4982.5  322.78  4989.2  323.48    4994  327.52  5024.6  330.72  5072.3  322.12
  5072.8  321.62    5090  322.12  5090.3   322.3  5095.3  325.26  5123.6  331.35
  5233.2  331.95  5286.8  333.76  5477.1  338.72  5862.2  340.39  6165.4  342.96
  6195.1  343.72  6424.7  347.85  6542.6  352.54  6608.5  363.72  6693.4  365.49
#Mann= 11 ,-1 , 0
  4323.6     .07       0    4994     .12       0  5072.3     .05       0
    5090     .12       0  5090.3      .1       0  5233.2     .12       0
  5286.8     .07       0  5862.2     .05       0  6165.4     .07       0
  6195.1     .05       0  6542.6     .07       0
Bank Sta=5072.3,5090
XS Rating Curve= 0 ,0
Exp/Cntr=0.3,0.1

Type RM Length L Ch R = 1 ,40584   ,464,464,464
BEGIN DESCRIPTION:
MOUND CREEK 56.0
END DESCRIPTION:
XS GIS Cut Line= 3
      2394124.97     13612424.97        2394725.       13613025.
        2395825.       13614125.
#Sta/Elev= 30
  4146.7  361.07  4203.3  357.92  4252.8  348.63    4274  346.48  4387.2  338.59
    4670  331.72  4945.8  331.93  4998.8  328.15  5000.5     321    5001   320.5
  5018.3     321  5023.6  325.37  5037.7  330.63  5094.3  330.71  5136.7  328.09
  5193.3  332.01  5278.1  331.42  5292.3  329.86  5351.5  333.95  5447.8   337.1
  5546.8  337.85  5631.7  334.77  5730.7  338.86  6041.8  341.95  6210.7   346.1
  6381.2  353.64  6437.8  359.18  6466.1  365.13  6494.3  373.78  6550.9   375.9
#Mann= 6 ,-1 , 0
  4146.7     .07       0  4945.8     .12       0  5000.5     .05       0
  5018.3     .12       0  5351.5     .05       0  6210.7    .035       0
Bank Sta=5000.5,5018.3
XS Rating Curve= 0 ,0
Exp/Cntr=0.3,0.1

Type RM Length L Ch R = 1 ,40120   ,517,517,517
BEGIN DESCRIPTION:
MOUND CREEK 55.0
END DESCRIPTION:
XS GIS Cut Line= 3
      2394075.02     13612875.02        2394675.       13613475.
      2395225.03     13613875.02
#Sta/Elev= 30
    4151  342.64  4179.2  341.78    4250  337.31  4405.5  333.73  4518.7  333.08
  4532.8  333.95  4561.1  332.83  4730.4  333.32  4744.9  333.43  4815.6  328.69
  4843.9  330.18  4893.4  331.02  4971.2  330.23  4985.4  328.35    4987  321.42
  4987.5  320.92  5004.9  321.42    5013  323.76  5021.5  328.66  5042.4  328.94
    5086  334.54  5142.8  334.98  5172.2  333.73  5199.5   334.4  5324.9  335.75
  5450.4  336.79  5557.1  340.75  5607.4  344.59  5642.9  348.14  5679.6  349.73
#Mann= 7 ,-1 , 0
    4151     .07       0  4730.4      .1       0    4987     .05       0
  5004.9      .1       0  5199.5     .07       0  5324.9     .05       0
  5607.4    .035       0
Bank Sta=4987,5004.9
XS Rating Curve= 0 ,0
Exp/Cntr=0.3,0.1

Type RM Length L Ch R = 1 ,39603   ,426,426,426
BEGIN DESCRIPTION:
B19632
END DESCRIPTION:
XS GIS Cut Line= 4
      2393801.39     13612963.62      2393997.03     13613442.96
      2394495.94     13613873.38      2395395.97     13614254.92
#Sta/Elev= 30
  4014.9  355.06    4273   347.2  4502.4  334.12  4683.6  331.18  4773.7  329.85
  4943.7  332.33    4979  326.59  4993.1  328.77  5000.7  326.72    5006  318.33
  5006.5  317.83    5024  318.33  5029.2  327.28  5035.8  328.83  5118.1  329.31
    5185  328.73  5201.4  331.91  5213.1  337.54  5231.3  336.82  5244.8  330.82
  5260.4  329.93  5413.3  330.15    5478  333.44  5567.7  334.85  5580.9  335.08
  5748.2  338.32  5865.9  345.47  5893.6   346.7  6157.6  347.73  6169.1  348.03
#Mann= 11 ,-1 , 0
  4014.9     .07       0  4683.6     .12       0    5006     .05       0
    5024     .12       0  5118.1      .1       0    5478     .07       0
  5567.7    .035       0  5580.9     .07       0  5865.9     .12       0
  5893.6     .07       0  6157.6     .12       0
Bank Sta=5006,5024
XS Rating Curve= 0 ,0
Exp/Cntr=0.3,0.1

Type RM Length L Ch R = 1 ,39177   ,369,369,369
BEGIN DESCRIPTION:
MOUND CREEK 54.0
END DESCRIPTION:
XS GIS Cut Line= 3
      2393145.96     13613550.56      2394398.11     13614117.94
      2395160.59     13614518.73
#Sta/Elev= 30
  3650.2  343.58  3763.2  343.73  4130.1  339.89  4399.6  332.92  4401.1   332.9
  4446.8  331.82  4521.5  326.26  4604.3   329.5    4637  329.19  4703.1  324.93
  4711.8   328.2  4725.1  329.78    4780   331.6  4865.8   328.4  4982.2   327.5
  4999.5  319.84  5001.8  316.94  5002.3  316.44  5019.8  316.94  5020.5  323.85
  5033.8  326.47  5094.5  330.93    5204  331.66  5221.5  331.53  5313.5  332.42
  5485.5   336.1  5540.3  339.02  5612.1  339.57  5760.7  346.13  5886.3  348.31
#Mann= 11 ,-1 , 0
  3650.2     .07       0  3763.2     .12       0  4399.6     .07       0
  4401.1     .12       0  4865.8      .1       0  5001.8     .05       0
  5019.8      .1       0  5094.5     .12       0    5204     .07       0
  5221.5     .12       0  5313.5     .07       0
Bank Sta=5001.8,5019.8
XS Rating Curve= 0 ,0
Exp/Cntr=0.3,0.1

Type RM Length L Ch R = 1 ,38808   ,435,435,435
BEGIN DESCRIPTION:
MOUND CREEK 53.0
END DESCRIPTION:
XS GIS Cut Line= 3
      2393625.03     13614225.01        2394225.       13614425.
      2394824.97     13614674.99
#Sta/Elev= 30
  4371.7  337.73  4508.7  332.68  4540.3  330.02  4561.4  330.65  4645.7  323.38
  4656.3  320.36  4677.4  325.64    4709  328.37  4729.8  328.48  4772.2  328.03
  4803.9  325.22  4888.2  326.26  4909.3  327.78  4930.3  326.32    4962  326.47
  4972.5   324.8    4974  316.45  4974.5  315.95    4992  316.45  4993.6  321.23
  5001.5   329.5  5013.3   330.4  5101.6  331.09  5223.5  329.97  5246.9  329.91
  5401.2  330.89  5485.7  334.86  5514.9  337.53  5556.6  338.82  5654.1  345.27
#Mann= 7 ,-1 , 0
  4371.7     .12       0  4729.8      .1       0    4974     .05       0
    4992      .1       0  5223.5     .07       0  5246.9     .12       0
  5401.2     .07       0
Bank Sta=4974,4992
XS Rating Curve= 0 ,0
Exp/Cntr=0.3,0.1

Type RM Length L Ch R = 1 ,38373   ,462,462,462
BEGIN DESCRIPTION:
MOUND CREEK 52.0
END DESCRIPTION:
XS GIS Cut Line= 3
      2393067.75     13614362.52        2393875.       13614575.
      2394874.95     13614774.99
#Sta/Elev= 30
  4165.3  339.57  4166.9  339.64    4275   339.5  4462.3  340.82  4589.6   339.4
  4658.8  335.49  4679.5  336.77  4731.2  333.51  4751.9  329.92  4793.2  327.71
    4907  328.21  4927.7  324.88  4936.5  325.08  4942.1  326.47  4977.3  323.62
  4980.6   315.2  4981.1   314.7  4998.8   315.2    5000  317.05  5002.6  317.05
  5010.2  324.74  5020.4  327.09  5081.6   326.1  5186.3  328.53  5538.5  329.05
  5673.1  330.24  5764.9  334.34  5877.1  340.76  5958.7  350.49  6019.8  352.43
#Mann= 8 ,-1 , 0
  4165.3     .12       0  4166.9    .033       0    4275     .12       0
  4936.5      .1       0  4980.6     .05       0  4998.8      .1       0
  5186.3     .12       0  5538.5     .07       0
Bank Sta=4980.6,4998.8
XS Rating Curve= 0 ,0
Exp/Cntr=0.3,0.1

Type RM Length L Ch R = 1 ,37911   ,468,468,468
BEGIN DESCRIPTION:
MOUND CREEK 51.0
END DESCRIPTION:
XS GIS Cut Line= 3
      2393474.99       13614875.        2393825.       13614925.
        2394925.       13614825.
#Sta/Elev= 30
  4641.6  335.81  4813.3  331.04  4914.4  325.06  4944.7  325.15  4964.9  323.79
  4978.1  325.39  4985.1  325.58  4997.7   324.2  5005.2  316.28  5006.1  314.43
  5006.6  313.93  5024.4  314.43  5025.3  321.98  5035.3   325.4  5055.4  326.41
  5105.6  325.52  5135.7  327.28    5171  327.28  5216.1  324.76  5336.6  326.26
  5365.9  327.37  5406.9   328.1  5457.1  327.55  5477.1  326.37  5527.3  328.41
  5587.6  328.35  5708.1  330.98  5798.5  334.74  5989.2  347.85  6099.7  353.67
#Mann= 6 ,-1 , 0
  4641.6     .12       0  4978.1      .1       0  5006.1     .05       0
  5024.4      .1       0    5171     .12       0  5365.9     .07       0
Bank Sta=5006.1,5024.4
XS Rating Curve= 0 ,0
Exp/Cntr=0.3,0.1

Type RM Length L Ch R = 1 ,37443   ,465,465,465
BEGIN DESCRIPTION:
MOUND CREEK 50.0
END DESCRIPTION:
XS GIS Cut Line= 3
        2393425.       13615025.        2393875.       13615375.
      2394775.01       13615375.
#Sta/Elev= 30
  4429.9  334.13    4564  331.07  4607.3  329.73  4657.9  326.01  4700.5  326.12
  4743.9  321.57    4772  325.42  4832.7  324.53  4907.7  326.27  4949.3  325.01
  4957.5  323.25  4971.9  315.07  4978.3  320.49  4987.6  313.66  4988.1  313.16
  5006.1  313.66    5010  314.89    5020  320.91    5030   323.1    5080  323.73
    5090  325.11  5155.8  324.76    5420  327.69  5618.7  327.73    5690  328.06
    5740   329.9    5840  338.12    5860  340.45    5890  346.59    5900  347.05
#Mann= 7 ,-1 , 0
  4429.9     .07       0    4564     .12       0  4832.7      .1       0
  4987.6     .05       0  5006.1      .1       0  5155.8     .07       0
  5618.7      .1       0
Bank Sta=4987.6,5006.1
XS Rating Curve= 0 ,0
Exp/Cntr=0.3,0.1

Type RM Length L Ch R = 1 ,36978   ,422,422,422
BEGIN DESCRIPTION:
MOUND CREEK 49.0
END DESCRIPTION:
XS GIS Cut Line= 3
      2393324.95       13615775.        2393825.       13615825.
      2394924.96       13615825.
#Sta/Elev= 30
  4492.8  334.23  4693.8     329  4834.5  321.56  4854.6  321.65  4884.8  323.36
  4927.4  322.31  4947.6  322.23  4975.2  323.96  4997.8  323.55  5005.3  319.48
  5015.3  315.53  5016.1  313.31  5016.6  312.81  5034.6  313.31  5045.3  317.15
  5055.3  324.86  5105.3  324.97  5194.6  323.58  5286.5  323.02  5345.3  320.99
  5384.9  320.95  5495.3  325.56  5735.3  326.22  5765.3  326.97  5789.8  328.88
  5875.1  336.87  5925.3  342.44  5955.3  344.61  6087.5  349.06  6095.3   349.2
#Mann= 10 ,-1 , 0
  4492.8     .12       0  4927.4      .1       0  5016.1     .05       0
  5034.6      .1       0  5194.6     .07       0  5286.5     .12       0
  5384.9     .07       0  5789.8     .12       0  5875.1     .07       0
  6087.5     .05       0
Bank Sta=5016.1,5034.6
XS Rating Curve= 0 ,0
Exp/Cntr=0.3,0.1

Type RM Length L Ch R = 1 ,36556   ,1121,1121,1121
BEGIN DESCRIPTION:
MOUND CREEK 48.0
END DESCRIPTION:
XS GIS Cut Line= 3
      2393375.01     13615975.01        2393825.       13616175.
        2394925.       13615875.
#Sta/Elev= 30
  4514.3  331.75  4696.9  328.55    4766  317.72  4772.1   321.5  4870.6  320.93
  4876.1     324  4885.2  319.65  4893.9  312.16  4899.3  318.13  4908.2   312.4
  4917.1  312.12  4922.6  317.35  4940.4  313.31    4952  316.81  4969.1   312.4
  4974.6  316.01  4991.5  312.57  4994.6  311.03  4995.1  310.53  5013.3  311.03
    5024  321.34  5048.2  322.94    5411  320.75  5431.7  317.06  5599.3  324.69
  5711.5   325.5  5877.4  330.46  5936.1  342.16  5972.4  343.63  6146.9  349.85
#Mann= 7 ,-1 , 0
  4514.3     .12       0  4885.2     .07       0  4991.5      .1       0
  4994.6     .05       0  5013.3      .1       0  5711.5     .12       0
  5972.4     .07       0
Bank Sta=4994.6,5013.3
XS Rating Curve= 0 ,0
Exp/Cntr=0.3,0.1

Type RM Length L Ch R = 1 ,35435   ,646,646,646
BEGIN DESCRIPTION:
MOUND CREEK 47.0
END DESCRIPTION:
XS GIS Cut Line= 3
      2393274.96     13616825.02      2394212.25     13616436.38
      2394975.25     13616005.97
#Sta/Elev= 30
  3567.9  338.69  3727.4  333.81  4141.7  324.36  4304.1   321.3  4370.7  321.59
  4411.7  321.69  4423.2  318.22  4446.4  321.44  4511.2  321.12  4872.8  320.22
  4917.1  319.31  4930.2  317.22  4953.1  319.96  4960.4  318.17  4966.1  319.78
  4982.1  318.41  5003.7  319.53    5016  310.36  5016.5  309.86  5034.7  310.36
  5041.3  318.18  5047.9  320.37  5062.9  326.45  5078.9  328.25  5194.2   333.8
  5246.4  340.17  5305.6  344.88  5370.6  348.14  5450.6  349.01  5458.6  349.25
#Mann= 8 ,-1 , 0
  3567.9     .07       0  3727.4     .05       0  4370.7     .07       0
  4511.2      .1       0    5016     .05       0  5034.7      .1       0
  5047.9     .07       0  5450.6     .05       0
Bank Sta=5016,5034.7
XS Rating Curve= 0 ,0
Exp/Cntr=0.3,0.1

Type RM Length L Ch R = 1 ,34789   ,437,437,437
BEGIN DESCRIPTION:
MOUND CREEK 46.0
END DESCRIPTION:
XS GIS Cut Line= 3
      2393674.99       13617125.        2394275.       13616725.
      2394874.98     13616475.01
#Sta/Elev= 30
  4272.6  330.85  4286.1  330.15  4301.2  330.77  4367.3  327.54  4380.8  328.35
  4409.3  326.56  4488.9  325.64  4625.7  322.36  4844.4  321.01    4872  321.05
  4893.1  322.34  4973.9  318.81  4996.4  317.36  5002.9  313.07    5006  309.85
  5006.5  309.35  5024.8  309.85  5032.2  315.04  5047.9  317.82  5102.1  321.77
  5114.5  322.41  5132.9   320.9  5156.2  321.81  5229.6  322.29  5330.4  323.72
  5357.9  324.33  5492.1  327.57  5581.4  332.11  5611.2  334.52  5643.7  335.68
#Mann= 8 ,-1 , 0
  4272.6     .05       0  4844.4     .07       0  4973.9      .1       0
    5006     .05       0  5024.8      .1       0  5229.6     .07       0
  5330.4      .1       0  5357.9     .07       0
Bank Sta=5006,5024.8
XS Rating Curve= 0 ,0
Exp/Cntr=0.3,0.1

Type RM Length L Ch R = 1 ,34352   ,445,445,445
BEGIN DESCRIPTION:
MOUND CREEK 45.0
END DESCRIPTION:
XS GIS Cut Line= 3
        2393775.       13617475.        2394375.       13617125.
      2394974.97     13616525.03
#Sta/Elev= 30
  4309.6   332.4  4403.5  329.56  4434.9  329.71  4440.7  328.71  4483.7   328.1
  4668.5  321.46  4749.5  319.52  4851.6  321.18  4937.6  319.63  4959.1  317.28
  4969.1  313.66  4971.7  310.63  4972.2  310.13  4990.5  310.63  4996.4  313.12
  5001.3  317.28  5018.4  318.44  5089.1  318.06    5116  318.83  5146.5  319.83
  5216.3  321.73  5329.5   321.2  5470.9  322.93    5485  321.79  5499.2  323.47
  5598.2   325.5  5668.9  328.45  5711.3  333.59  5810.3  339.06  5852.7  342.51
#Mann= 5 ,-1 , 0
  4309.6     .07       0  4971.7     .05       0  4990.5     .07       0
    5116      .1       0  5146.5     .07       0
Bank Sta=4971.7,4990.5
XS Rating Curve= 0 ,0
Exp/Cntr=0.3,0.1

Type RM Length L Ch R = 1 ,33907   ,447,447,447
BEGIN DESCRIPTION:
MOUND CREEK 44.0
END DESCRIPTION:
XS GIS Cut Line= 3
      2393924.98     13617675.01        2394525.       13617525.
      2395124.99     13617025.01
#Sta/Elev= 30
  4381.1  330.68  4432.7  329.64  4522.9  325.54    4680  322.03    4729  319.69
  4816.6  319.46  4875.9  317.45  4893.9  315.13  4899.1  317.23  4946.7   317.9
  4968.7   315.7  4976.4  312.84  4979.9  309.57  4980.4  309.07  4998.7  309.57
  4999.6  310.47  5002.8  310.47  5006.8  314.01  5013.3  312.88  5021.1  316.46
  5189.2  319.96  5390.1  319.48  5481.9  321.38  5510.5  322.65  5588.6  328.68
  5617.3  328.82  5666.7  331.86    5724  336.77  5759.1  341.95  5780.6  343.26
#Mann= 5 ,-1 , 0
  4381.1     .07       0  4946.7      .1       0  4979.9     .05       0
  4998.7      .1       0  5189.2     .07       0
Bank Sta=4979.9,4998.7
XS Rating Curve= 0 ,0
Exp/Cntr=0.3,0.1

Type RM Length L Ch R = 1 ,33460   ,468,468,468
BEGIN DESCRIPTION:
MOUND CREEK 43.0
END DESCRIPTION:
XS GIS Cut Line= 3
      2394275.01     13618474.99        2394725.       13617875.
      2395275.01     13617374.99
#Sta/Elev= 30
  4249.6  334.89    4586   323.7  4842.3  319.31  4927.7  315.98  4948.5  316.44
  4968.3  314.53  4971.5  313.47  4976.6  308.78  4977.1  308.28  4995.5  308.78
  4996.5   310.3    5003   310.3  5006.7  313.24  5013.4  315.41  5020.9  316.38
  5070.2     317  5134.4  315.93  5155.3  314.34  5169.5  316.28  5221.5  318.41
  5301.2  318.35  5306.2  318.34  5437.8  319.27  5574.3  323.34  5643.9  330.72
  5672.3  336.77    5679  339.22  5700.7  342.73  5717.8  343.69  5742.9  345.04
#Mann= 10 ,-1 , 0
  4249.6     .07       0  4948.5      .1       0  4976.6     .05       0
  4995.5      .1       0  5221.5     .07       0  5301.2    .035       0
  5306.2     .07       0  5437.8    .063       0  5574.3     .07       0
  5717.8     .12       0
Bank Sta=4976.6,4995.5
XS Rating Curve= 0 ,0
Exp/Cntr=0.3,0.1

Type RM Length L Ch R = 1 ,32992   ,472,472,472
BEGIN DESCRIPTION:
MOUND CREEK 42.0
END DESCRIPTION:
XS GIS Cut Line= 3
      2394725.01     13618424.99        2395075.       13618125.
      2395375.01     13617524.99
#Sta/Elev= 30
  4544.3  326.61  4683.4  322.81  4721.5  321.21  4728.7  318.83  4735.8  319.93
  4764.4  318.29  4778.6  319.34  4785.2  317.58  4792.9  319.13  4816.3  317.66
  4856.5  315.54  4945.9  314.45  4949.2  314.54    4963  314.73  4977.3  306.59
    4982  305.56  4982.5  305.06    5001  305.56    5002  313.51  5008.1  313.51
  5013.7  315.34  5080.7  314.03  5117.1  316.92  5184.2  317.92  5319.7  316.33
  5452.5  319.62  5527.9  323.85  5600.6  330.33  5656.2  340.31  5676.1  341.11
#Mann= 9 ,-1 , 0
  4544.3     .07       0  4683.4    .035       0  4816.3     .07       0
  4945.9    .035       0  4949.2      .1       0    4982     .05       0
    5001      .1       0  5319.7     .07       0  5656.2     .12       0
Bank Sta=4982,5001
XS Rating Curve= 0 ,0
Exp/Cntr=0.3,0.1

Type RM Length L Ch R = 1 ,32520   ,438,438,438
BEGIN DESCRIPTION:
MOUND CREEK 41.0
END DESCRIPTION:
XS GIS Cut Line= 3
      2395174.98     13618825.04        2395425.       13618375.
      2395924.98     13618075.01
#Sta/Elev= 30
  4491.3  330.49  4537.1  329.16  4689.2  318.65  4823.1  315.63  4835.7  314.06
  4850.5  313.74  4873.4  311.86  4903.2  313.32  4916.9  312.72  4960.4  313.95
  4970.7   313.4  4976.4  306.96  4982.8  302.61  4983.3  302.11    5002  302.61
  5003.3  304.12    5009  304.12  5019.7  309.84  5041.1  315.09  5099.4  314.62
  5135.6  315.47  5181.1  316.04  5225.8  318.56    5253  318.83  5274.3  320.14
  5342.4  320.96  5348.2  321.81  5363.8  321.03  5464.8  321.25  5589.2  322.46
#Mann= 5 ,-1 , 0
  4491.3     .07       0  4850.5      .1       0  4982.8     .05       0
    5002      .1       0  5135.6     .07       0
Bank Sta=4982.8,5002
XS Rating Curve= 0 ,0
Exp/Cntr=0.3,0.1

Type RM Length L Ch R = 1 ,32082   ,449,449,449
BEGIN DESCRIPTION:
MOUND CREEK 40.0
END DESCRIPTION:
XS GIS Cut Line= 3
      2395425.02     13619024.98        2395675.       13618725.
      2395774.99     13618475.04
#Sta/Elev= 30
    4603  331.27  4624.4  330.14  4638.8  328.39  4666.7  321.95  4673.9   319.7
  4709.1  315.67  4759.2  313.82    4795  313.94  4806.7  313.16  4845.5  312.41
  4879.6  312.13  4887.4  311.37    4929  312.79  4943.4  309.85  4979.8  311.88
  4986.3  310.26  4990.2  307.23  4996.2  307.23  4998.7  300.28  4999.2  299.78
  5017.9  300.28  5025.8  304.78  5032.5   309.9  5037.9  312.19  5062.1  313.42
  5068.9  316.22  5079.6  318.04  5101.2  319.29  5253.4     321  5262.7  320.93
#Mann= 7 ,-1 , 0
    4603     .07       0  4666.7     .12       0  4806.7     .07       0
  4845.5      .1       0  4998.7     .05       0  5017.9      .1       0
  5253.4     .07       0
Bank Sta=4998.7,5017.9
XS Rating Curve= 0 ,0
Exp/Cntr=0.3,0.1

Type RM Length L Ch R = 1 ,31633   ,453,453,453
BEGIN DESCRIPTION:
MOUND CREEK 39.0
END DESCRIPTION:
XS GIS Cut Line= 3
        2395425.       13619125.        2395975.       13619025.
        2396425.       13618675.
#Sta/Elev= 30
  4436.3  333.47    4463  333.59    4477  332.54  4516.3  326.85  4521.4   327.6
  4527.8  325.08  4548.3  322.15  4639.6  314.71  4700.6  311.72  4759.3  310.78
  4822.5   310.2  4893.7  312.14  4934.3  310.52  5002.6  311.82  5007.4   299.6
  5007.9   299.1  5026.7   299.6  5031.5  299.72  5037.8  302.67    5046  301.73
  5058.7  306.52  5073.1  307.93  5081.3  310.34  5095.8  311.93  5116.6  311.46
  5223.1  314.33  5333.9  316.51  5379.9  316.66  5520.5  319.83  5565.4  320.49
#Mann= 8 ,-1 , 0
  4436.3     .07       0  4548.3     .12       0  4759.3      .1       0
  5007.4     .05       0  5026.7      .1       0  5223.1     .07       0
  5333.9     .12       0  5520.5     .07       0
Bank Sta=5007.4,5026.7
XS Rating Curve= 0 ,0
Exp/Cntr=0.3,0.1

Type RM Length L Ch R = 1 ,31180   ,438,438,438
BEGIN DESCRIPTION:
MOUND CREEK 38.0
END DESCRIPTION:
XS GIS Cut Line= 3
      2395424.98       13619225.        2396225.       13619325.
      2396575.02     13618824.98
#Sta/Elev= 30
  4193.8  332.96  4236.7  331.92  4304.7  327.52  4382.6  319.35  4405.5  317.03
  4536.5   313.3  4634.7  308.18  4677.6  307.89  4788.4  310.74    4859  309.38
  4939.6  311.11  4949.7  301.52  4954.3  300.15  4957.2  299.28  4962.3  305.86
  4969.8  302.03  5003.1  300.37  5003.9  299.11  5004.4  298.61  5023.2  299.11
  5028.4  300.12  5036.7  304.19    5058  308.47  5064.1  311.79    5096  311.23
  5169.4  312.18  5344.6  316.36  5364.5  316.61  5561.9  319.34  5610.4  320.39
#Mann= 10 ,-1 , 0
  4193.8     .07       0  4382.6     .12       0  4954.3      .1       0
  5003.9     .05       0  5023.2      .1       0    5096     .12       0
  5169.4     .07       0  5344.6     .12       0  5364.5     .07       0
  5561.9     .12       0
Bank Sta=5003.9,5023.2
XS Rating Curve= 0 ,0
Exp/Cntr=0.3,0.1

Type RM Length L Ch R = 1 ,30742   ,435,435,435
BEGIN DESCRIPTION:
MOUND CREEK 37.0
END DESCRIPTION:
XS GIS Cut Line= 3
        2395575.       13619525.        2396175.       13619675.
      2396875.01       13619275.
#Sta/Elev= 30
  4374.5  320.33  4907.7   307.9    4962   308.9  4990.4  298.85  5000.9  300.97
  5044.1  298.39  5059.9  304.15  5065.7  301.39  5081.5  309.13  5087.3  304.19
  5096.6   309.5  5103.1  310.08  5108.9  305.94  5118.9  307.91  5124.7  301.93
  5136.3  298.14  5136.8  297.64  5156.2  298.14  5162.1  304.48  5167.9  298.47
  5183.7  310.61  5323.4  308.15  5338.5  311.15    5463  311.33  5468.8  305.05
  5484.6  305.05  5490.4  309.43    5512  312.38  5576.2  312.87  5799.2  321.81
#Mann= 5 ,-1 , 0
  4374.5     .07       0  4907.7      .1       0  5136.3     .05       0
  5156.2      .1       0  5576.2     .12       0
Bank Sta=5136.3,5156.2
XS Rating Curve= 0 ,0
Exp/Cntr=0.3,0.1
