--- SHOCKLEY CREEK.prj (project) ---

Proj Title=SHOCKLEY CREEK Base Level Engineering
Current Plan=p01
Default Exp/Contr=0.3,0.1
English Units
Geom File=g01
Flow File=f01
Plan File=p01
Y Axis Title=Elevation
X Axis Title(PF)=Main Channel Distance
X Axis Title(XS)=Station
BEGIN DESCRIPTION:
SHOCKLEY CREEK
END DESCRIPTION:
DSS Export Rating Curves= 0
DSS Export Rating Curve Sorted= 0
DSS Export Volume Flow Curves= 0
DXF OffsetX= 0
DXF OffsetY= 0
DXF ScaleX= 1
DXF ScaleY= 10

--- SHOCKLEY CREEK.p01 (plan) ---

Plan Title=Multiple Run
Program Version=4.10
Short Identifier=Multiple
Geom File=g01
Flow File=f01
Subcritical Flow
K Sum by GR= 0
Std Step Tol= 0.01
Critical Tol= 0.01
Num of Std Step Trials= 20
Max Error Tol= 0.3
Flow Tol Ratio= 0.001
Split Flow NTrial= 30
Split Flow Tol= 0.02
Split Flow Ratio= 0.02
Log Output Level= 0
Friction Slope Method= 1
Unsteady Friction Slope Method= 2
Unsteady Bridges Friction Slope Method= 1
Parabolic Critical Depth
Global Vel Dist= 1 , 1 , 1
Global Log Level= 0
CheckData=True
Encroach Param=-1 ,0,0, 0
BEGIN DESCRIPTION:
Multiple Run
END DESCRIPTION:
Computation Interval=1HOUR
Output Interval=1HOUR
Run HTab= 0
Run UNet= 0
Run PostProcess= 0
Run WQNet= 0
UNET Theta= 1
UNET Theta Warmup= 1
UNET ZTol= 0.02
UNET ZSATol= 0.05
UNET MxIter= 20
UNET MaxInSteps= 0
UNET DtIC= 0
UNET DtMin= 0
UNET MaxCRTS= 20
UNET WFStab= 2
UNET SFStab= 1
UNET WFX= 1
UNET SFX= 1
UNET DSS MLevel= 4
UNET DZMax Abort= 100
UNET Convert EG Bridges= 0
UNET Use Existing IB Tables=-1
UNET Froude Reduction=False
UNET Froude Limit= 1
UNET Froude Power= 10
UNET Time Slicing=0,0, 5
UNET Junction Losses=0
Instantaneous Interval=1HOUR
Write IC File= 0
Write IC File at Sim End=0
Echo Input=False
Echo Parameters=False
Echo Output=False
Write Detailed= 0
WQ AD Non Conservative
WQ ULTIMATE=-1
WQ Max Comp Step=1HOUR
WQ Output Interval=15MIN
WQ Output Selected Increments= 0
WQ Output face flow=0
WQ Output face velocity=0
WQ Output face area=0
WQ Output face dispersion=0
WQ Output cell volume=0
WQ Output cell surface area=0
WQ Output cell continuity=0
WQ Output cumulative cell continuity=0
WQ Output face conc=0
WQ Output face dconc_dx=0
WQ Output face courant=0
WQ Output face peclet=0
WQ Output face adv mass=0
WQ Output face disp mass=0
WQ Output cell mass=0
WQ Output cell source sink temp=0
WQ Output cell source sink nsm=0
WQ Output MaxMinRange=-1
WQ Daily Max Min Mean=-1
WQ Daily Range=0
WQ Daily Time=0
WQ Create Restart=0
WQ Fixed Restart=0
WQ System Summary=0
WQ Use Fixed Temperature=0
Sorting and Armoring Iterations= 10
XS Update Threshold= 0.02
Hydraulics Update Threshold= 0.02
Energy Slope Method= 1
Volume Change Method= 0
XS Weighting Method= 0
Number of US Weighted Cross Sections= 1
Number of DS Weighted Cross Sections= 1
Upstream XS Weight=0.25
Main XS Weight=0.5
Downstream XS Weight=0.25
Number of DS XS's Weighted with US Boundary= 1
Upstream Boundary Weight= 1
Weight of XSs Associated with US Boundary= 0
Number of US XS's Weighted with DS Boundary= 1
Downstream Boundary Weight= 0.5
Weight of XSs Associated with DS Boundary= 0.5
Sediment Output Level= 4
Mass or Volume Output= 0
Output Increment Type= 1
Profile and TS Output Increment= 10
XS Output Flag= 0
XS Output Increment= 10
Disregard all LS=0
Disregard all Conn=0
Disregard all Breaches=0
Disregard all Pumps=0

--- SHOCKLEY CREEK.f01 (steady flow) ---

Flow Title=Multiple
Number of Profiles=7
Profile Names=10-year,25-year,50-year,1pct_min,100-year,1pct_plu,500-year
River Rch & RM= SHOCKLEY CREEK,Reach-1,25927
     766    1259    1711    1125    2244    4477    3829
River Rch & RM= SHOCKLEY CREEK,Reach-1,24144
    1105    1842    2527    1675    3341    6667    5798
River Rch & RM= SHOCKLEY CREEK,Reach-1,22758
    1264    2112    2902    1925    3840    7663    6674
River Rch & RM= SHOCKLEY CREEK,Reach-1,17298
    1937    3291    4571    3061    6107   12185   10820
River Rch & RM= SHOCKLEY CREEK,Reach-1,14971
    2201    3744    5203    3483    6950   13868   12310
River Rch & RM= SHOCKLEY CREEK,Reach-1,9076
    2308    3927    5462    3658    7298   14561   12933
River Rch & RM= SHOCKLEY CREEK,Reach-1,6874
    2351    3990    5538    3700    7383   14730   13023
Boundary for River Rch & Prof#=SHOCKLEY CREEK,Reach-1,1
Up Type=0
Dn Type=3
Dn Slope=0.005
Boundary for River Rch & Prof#=SHOCKLEY CREEK,Reach-1,2
Up Type=0
Dn Type=3
Dn Slope=0.005
Boundary for River Rch & Prof#=SHOCKLEY CREEK,Reach-1,3
Up Type=0
Dn Type=3
Dn Slope=0.005
Boundary for River Rch & Prof#=SHOCKLEY CREEK,Reach-1,4
Up Type=0
Dn Type=3
Dn Slope=0.005
Boundary for River Rch & Prof#=SHOCKLEY CREEK,Reach-1,5
Up Type=0
Dn Type=3
Dn Slope=0.005
Boundary for River Rch & Prof#=SHOCKLEY CREEK,Reach-1,6
Up Type=0
Dn Type=3
Dn Slope=0.005
Boundary for River Rch & Prof#=SHOCKLEY CREEK,Reach-1,7
Up Type=0
Dn Type=3
Dn Slope=0.005

--- SHOCKLEY CREEK.g01 (geometry) ---

Geom Title=Existing Conditions
Program Version=4.10

River Reach=SHOCKLEY CREEK  ,Reach-1
Reach XY= 30
        2351025.       13618925.      2353714.55     13619125.53
      2354209.75     13619575.55      2354799.88     13619224.68
      2355418.91     13619523.44      2355674.97     13619082.08
      2355985.25     13619474.03      2356185.43     13619225.53
      2356864.39     13619324.41      2357068.92     13618976.56
      2357222.42     13619870.05      2357823.78     13619728.43
      2358540.23     13620324.76      2359273.55     13620078.53
      2359422.56     13620719.61      2359823.58     13620578.04
       2360072.3     13620969.64      2361930.86     13621872.95
      2362581.08     13621783.13      2362698.13     13622698.85
      2363331.06     13622483.14      2364802.35     13623550.97
      2364680.05     13623877.28      2365149.48     13624047.84
      2365272.58     13624469.61      2365504.85     13623874.28
       2365817.4     13624121.66      2365771.65     13624617.41
      2366759.64     13624775.11        2367375.       13624425.

Type RM Length L Ch R = 1 ,25927   ,366,366,366
BEGIN DESCRIPTION:
E20828
END DESCRIPTION:
XS GIS Cut Line= 3
      2351085.98     13619673.28       2351131.7     13618861.69
      2351228.87     13618444.43
#Sta/Elev= 30
  4296.6  354.86  4425.1  353.48  4445.1  354.53  4455.1  353.11  4465.1  352.97
  4548.1  353.33  4685.5  351.89  4825.7  352.17  4855.8  350.05  4901.1  345.48
  4955.9  345.15    4976  344.12  4993.5   341.1  4993.8   340.6  4998.5   341.1
    5006  341.73    5016  344.77  5018.5  344.81    5036  346.15  5096.1  347.62
    5144  351.31  5149.2  350.25  5167.7  350.25  5191.7  351.56  5269.7  353.04
  5315.6  353.55  5403.8  354.99  5434.6  356.69  5479.2  357.52  5537.9  358.91
#Mann= 7 ,-1 , 0
  4296.6     .07       0  4993.5     .05       0  4998.5     .07       0
  5018.5      .1       0  5269.7     .07       0  5315.6    .035       0
  5479.2     .07       0
Bank Sta=4993.5,4998.5
XS Rating Curve= 0 ,0
Exp/Cntr=0.3,0.1

Type RM Length L Ch R = 1 ,25561   ,478,478,478
BEGIN DESCRIPTION:
SHOCKLEY CREEK 30.0
END DESCRIPTION:
XS GIS Cut Line= 3
      2351343.17     13619759.02        2351475.       13618925.
      2351524.99     13618675.03
#Sta/Elev= 30
  4155.6  354.65  4250.8  352.81  4259.6  353.09  4264.7  352.42  4341.9   351.5
  4372.3  351.78  4394.5  351.26  4483.6  351.12  4655.8  349.59  4711.6  349.93
  4797.5   349.6  4817.7  348.66  4836.4  348.36  4848.1  348.76  4915.6  347.31
  4929.1  346.72  4959.5  343.89  4971.3  343.61  4979.7  342.88  4989.9  341.44
  4994.9  338.08  4995.3  337.58  4999.6  337.58  4999.9  338.08  5002.5  338.08
  5010.2  343.49  5147.2  351.41  5173.3  351.99  5183.5  352.64  5254.9  354.06
#Mann= 5 ,-1 , 0
  4155.6     .07       0  4915.6      .1       0  4994.9     .05       0
  4999.9      .1       0  5147.2     .07       0
Bank Sta=4994.9,4999.9
XS Rating Curve= 0 ,0
Exp/Cntr=0.3,0.1

Type RM Length L Ch R = 1 ,25083   ,484,484,484
BEGIN DESCRIPTION:
SHOCKLEY CREEK 29.0
END DESCRIPTION:
XS GIS Cut Line= 3
        2351325.       13619925.        2351875.       13619125.
        2351875.     13618675.02
#Sta/Elev= 30
  4029.7  358.44  4087.9  357.23  4187.5  354.03  4381.6  350.86  4512.1   350.3
  4661.6  347.79  4742.1  349.04  4777.9     349  4879.2  347.55  4936.3  348.01
  4957.2  346.42  4972.1  344.01  4978.2  345.88    4987   342.9  4993.1  343.49
  4997.5  340.81  5010.5  341.13    5018  338.32  5018.4  337.82  5022.7  337.82
  5023.1  338.32  5030.5  342.26  5065.4  342.64  5140.5  342.91  5180.5  343.97
  5220.5  345.94  5258.1  348.61  5290.5  350.13  5444.3  354.79  5450.5     355
#Mann= 6 ,-1 , 0
  4029.7     .07       0    5018     .05       0  5023.1     .07       0
  5065.4      .1       0  5258.1     .07       0  5444.3    .035       0
Bank Sta=5018,5023.1
XS Rating Curve= 0 ,0
Exp/Cntr=0.3,0.1

Type RM Length L Ch R = 1 ,24599   ,455,455,455
BEGIN DESCRIPTION:
SHOCKLEY CREEK 28.0
END DESCRIPTION:
XS GIS Cut Line= 3
      2352263.35     13619879.02        2352325.       13619125.
      2352223.34     13618541.63
#Sta/Elev= 30
  4247.6  349.62  4622.9  347.38  4697.7  345.79  4763.3  341.55  4783.4  341.54
  4819.3  339.39  4833.6  339.17  4843.6  340.61  4846.6  340.29  4853.6  339.55
  4893.8  344.29  4923.9  345.45    4954  343.62    4974   338.8  4999.1   338.4
  4999.5   337.9  5004.2   338.4  5014.3  338.58  5031.4     341  5054.9   342.6
    5096     344  5210.1  345.84  5278.2  348.19  5288.4  347.93  5308.7  345.52
  5324.2  348.67  5342.9  349.15  5443.5  351.72  5572.6  355.46  5596.3  355.51
#Mann= 6 ,-1 , 0
  4247.6     .07       0  4846.6      .1       0  4999.1     .05       0
  5004.2      .1       0  5342.9    .035       0  5443.5     .07       0
Bank Sta=4999.1,5004.2
XS Rating Curve= 0 ,0
Exp/Cntr=0.3,0.1

Type RM Length L Ch R = 1 ,24144   ,486,486,486
BEGIN DESCRIPTION:
SHOCKLEY CREEK 27.0
END DESCRIPTION:
XS GIS Cut Line= 3
      2352324.99     13619875.04        2352625.       13618975.
      2352524.98     13618674.95
#Sta/Elev= 30
  4056.3  349.31    4109  349.28  4657.2  345.06  4709.9  343.57    4731  341.49
  4762.6  340.54  4776.7  340.64  4846.9  339.47  4878.5   340.3  4920.7  339.66
    4926  340.39  4931.2  339.84  4938.2  334.18  4938.7  333.68  4944.8  333.68
  4945.3  334.18  4952.3  335.47  4973.4  336.49  4983.9  337.53  5002.4   340.2
  5007.7   340.2  5015.6  341.44  5026.1  341.51  5047.2  342.76  5056.2  342.06
  5089.4  342.24  5131.5  343.66  5163.1  346.43  5194.8  348.08  5321.3  352.14
#Mann= 5 ,-1 , 0
  4056.3     .07       0  4776.7      .1       0  4938.2     .05       0
  4945.3      .1       0  5056.2     .07       0
Bank Sta=4938.2,4945.3
XS Rating Curve= 0 ,0
Exp/Cntr=0.3,0.1

Type RM Length L Ch R = 1 ,23658   ,448,448,448
BEGIN DESCRIPTION:
SHOCKLEY CREEK 26.0
END DESCRIPTION:
XS GIS Cut Line= 3
      2352524.98     13619625.02        2352975.       13619175.
        2352925.     13618724.99
#Sta/Elev= 30
  4364.2  346.56  4463.2  345.71  4505.6     346  4590.5  344.42  4647.1  344.82
  4661.2  345.74  4675.4  344.68  4830.9  342.85  4868.3  341.36  4929.9  340.67
  4944.1  339.38  4958.2  334.44  4968.7  332.25  4969.2  331.75  4975.4  331.75
  4975.9  332.25  4986.5  336.84  5020.7  338.68  5050.9  338.57  5101.2  337.08
  5151.5  337.25  5161.6  337.88  5242.1  337.27  5282.3  338.87  5312.5  338.96
  5322.6  340.32  5352.8  341.75  5414.7  346.64  5433.3  348.64  5453.4  349.19
#Mann= 5 ,-1 , 0
  4364.2     .07       0  4868.3      .1       0  4968.7     .05       0
  4975.9      .1       0  5414.7     .07       0
Bank Sta=4968.7,4975.9
XS Rating Curve= 0 ,0
Exp/Cntr=0.3,0.1

Type RM Length L Ch R = 1 ,23210   ,452,452,452
BEGIN DESCRIPTION:
SHOCKLEY CREEK 25.0
END DESCRIPTION:
XS GIS Cut Line= 3
        2353375.     13619824.99        2353325.       13619175.
      2353075.01     13618525.03
#Sta/Elev= 30
  4348.8  345.68  4499.2  342.58  4632.5   342.3  4789.2  340.35  4890.4  335.86
  4940.5   338.8  4990.7  334.69  4994.6  329.27  4995.1  328.77  5001.8  329.27
  5015.7  330.92  5022.1   336.5    5065  335.28  5075.7  330.37  5086.4  332.03
    5095  330.92  5100.3  335.24  5107.8  329.98  5118.6  335.45    5215  335.04
  5378.9  337.44  5408.9  339.28    5440  345.06  5458.2  346.96  5506.4  347.42
  5572.8  350.01  5597.5  352.44  5622.1  351.03    5665  354.64  5697.1  354.87
#Mann= 6 ,-1 , 0
  4348.8     .07       0  4632.5      .1       0  4789.2     .07       0
  4994.6     .05       0  5001.8     .07       0  5506.4     .07       0
Bank Sta=4994.6,5001.8
XS Rating Curve= 0 ,0
Exp/Cntr=0.3,0.1

Type RM Length L Ch R = 1 ,22758   ,448,448,448
BEGIN DESCRIPTION:
SHOCKLEY CREEK 24.0
END DESCRIPTION:
XS GIS Cut Line= 3
        2353875.     13619925.01        2353725.       13619125.
        2353625.     13618324.98
#Sta/Elev= 30
  4190.2  350.81  4379.3  344.44  4736.5  339.25  4815.1  334.95  4831.2  333.06
  4837.7  328.75  4838.2  328.25  4845.1  328.75  4851.5  332.16  4867.6  333.69
  4872.7   331.5  4892.2  332.51  4902.4  329.23  4920.2  334.32  4972.8  335.53
  4983.8  335.41    4994  333.15  5001.6  329.43  5006.7  329.43  5024.3  335.46
  5041.9  338.77    5047  337.83  5059.1  339.34  5094.9  338.63  5387.1  342.18
  5558.4  346.31  5729.8  352.32  5749.9  354.09  5772.6  352.78  5810.4  355.19
#Mann= 5 ,-1 , 0
  4190.2     .07       0  4736.5      .1       0  4837.7     .05       0
  4845.1      .1       0  5059.1     .07       0
Bank Sta=4837.7,4845.1
XS Rating Curve= 0 ,0
Exp/Cntr=0.3,0.1

Type RM Length L Ch R = 1 ,22310   ,447,447,447
BEGIN DESCRIPTION:
SHOCKLEY CREEK 23.0
END DESCRIPTION:
XS GIS Cut Line= 3
        2353975.     13619674.97        2354025.       13619375.
        2353975.     13618574.97
#Sta/Elev= 30
  4696.2  343.32  4817.8  340.43  4872.6  339.93  4911.6  337.32  4967.4  336.91
  4990.2  334.07  4992.7  332.69  4997.8  329.87  5002.8  329.87  5006.6  327.99
  5007.1  327.49  5014.1  327.99  5020.4   331.9  5040.4  333.78  5150.6  333.05
  5190.7  331.46  5220.7  332.09  5238.3  333.37  5243.3  331.97  5290.9  333.54
    5351  331.81  5381.1  333.52  5441.2  335.25  5461.2  337.81  5475.2  338.68
  5501.3  338.02  5581.4  340.15  5601.5  341.52  5741.8   344.1  5801.9  346.23
#Mann= 6 ,-1 , 0
  4696.2     .07       0  4872.6     .12       0  4992.7      .1       0
  5006.6     .05       0  5014.1      .1       0  5475.2     .07       0
Bank Sta=5006.6,5014.1
XS Rating Curve= 0 ,0
Exp/Cntr=0.3,0.1

Type RM Length L Ch R = 1 ,21863   ,453,453,453
BEGIN DESCRIPTION:
SHOCKLEY CREEK 22.0
END DESCRIPTION:
XS GIS Cut Line= 3
        2354175.       13619725.        2354275.       13619575.
        2353975.     13618375.01
#Sta/Elev= 30
  4820.3  343.12  4908.4  341.51    4921  340.89    4951  334.53    4957  334.94
    4972  327.53  4987.1  330.12  4993.1   327.8  4997.6  331.91  5062.7  332.16
  5155.2  333.49  5299.5  332.54  5312.4  332.95  5348.5  341.07  5353.6  339.54
  5361.3  341.05  5389.7  339.49  5394.8  340.87  5430.9  332.43  5436.1   333.9
  5468.4  326.46  5468.9  325.96  5475.9  326.46  5577.8  330.93  5595.9  335.78
    5601   334.9  5637.1  339.11  5721.4  338.52  6054.5  346.08  6237.5  352.49
#Mann= 6 ,-1 , 0
  4820.3     .07       0  4908.4     .12       0  5062.7      .1       0
  5468.4     .05       0  5475.9      .1       0  5721.4     .07       0
Bank Sta=5468.4,5475.9
XS Rating Curve= 0 ,0
Exp/Cntr=0.3,0.1

Type RM Length L Ch R = 1 ,21410   ,433,433,433
BEGIN DESCRIPTION:
SHOCKLEY CREEK 21.0
END DESCRIPTION:
XS GIS Cut Line= 3
      2354825.01     13619975.05        2354675.       13619425.
      2354225.01     13618625.01
#Sta/Elev= 30
  4424.8  341.99  4435.2  342.97  4442.1  344.83  4447.3  343.02  4466.3  341.18
  4621.8  338.38  4642.5  336.99  4660.5  338.13  4669.8  337.89  4919.5  336.82
  4972.5  334.61  4977.7  332.18  4984.6  330.97  5002.9  330.16  5008.6  326.43
  5013.5  326.15    5014  325.65  5022.3  326.15  5024.6  326.29  5030.3  330.52
  5148.9  329.93  5235.9  336.16  5307.4  336.87  5332.4  337.43  5362.1  335.61
  5375.8  337.02  5409.7  337.24  5422.3  337.34  5721.3  338.13  5912.8  343.97
#Mann= 9 ,-1 , 0
  4424.8     .07       0  4660.5     .12       0  4669.8     .07       0
  4919.5      .1       0  5013.5     .05       0  5022.3      .1       0
  5307.4     .07       0  5409.7    .035       0  5422.3     .07       0
Bank Sta=5013.5,5022.3
XS Rating Curve= 0 ,0
Exp/Cntr=0.3,0.1

Type RM Length L Ch R = 1 ,20977   ,945,945,945
BEGIN DESCRIPTION:
SHOCKLEY CREEK 20.0
END DESCRIPTION:
XS GIS Cut Line= 3
      2355074.99     13619874.97        2354975.       13619275.
      2354225.02     13618475.02
#Sta/Elev= 30
    4374  339.86  4637.6  335.82  4691.9  333.61    4820  333.64    4873  331.69
  4982.2  329.31  4984.9   324.7  4985.4   324.2  4993.8   324.7  4996.2  329.25
  5003.5  324.89  5010.3   326.8  5024.5  325.79  5031.8  329.57  5038.7  328.18
    5046  329.75  5052.8  325.78  5060.1  328.35    5067  325.27  5074.3   327.8
  5081.2  326.52  5088.5  330.99    5114  332.66  5173.5  335.36  5194.5  335.26
  5208.6  333.35  5248.7  335.32  5528.7  336.45  5795.8  339.32  6078.8  347.37
#Mann= 8 ,-1 , 0
    4374     .07       0  4691.9     .12       0    4873      .1       0
  4984.9     .05       0  4993.8      .1       0    5114     .07       0
  5248.7    .035       0  5528.7     .07       0
Bank Sta=4984.9,4993.8
XS Rating Curve= 0 ,0
Exp/Cntr=0.3,0.1

Type RM Length L Ch R = 1 ,20032   ,457,457,457
BEGIN DESCRIPTION:
SHOCKLEY CREEK 19.0
END DESCRIPTION:
XS GIS Cut Line= 3
        2355625.     13619825.04        2355575.       13619275.
      2354774.98     13618474.98
#Sta/Elev= 30
  4460.5  339.25  4711.6  333.85  4731.7  332.88  4831.9  331.53  4842.1  331.47
  4882.3   327.9  4922.4  327.76  4942.5  323.84    4948   323.5  4948.5     323
  4957.1   323.5  4962.6  327.64  5055.2  327.53  5097.7  328.88  5125.9  331.73
  5167.5   332.3  5239.1   331.7  5281.5  329.83  5309.8  329.65  5338.1  331.59
  5366.4  330.13  5408.8  331.81  5465.4  332.03  5550.2  333.86  5720.2  335.12
  5726.3   335.2  5863.8   336.7  5946.2  337.07  6131.9  340.36  6144.2  340.81
#Mann= 9 ,-1 , 0
  4460.5     .07       0  4831.9      .1       0    4948     .05       0
  4957.1      .1       0  5167.5     .07       0  5720.2    .035       0
  5726.3     .07       0  5863.8    .035       0  6131.9     .05       0
Bank Sta=4948,4957.1
XS Rating Curve= 0 ,0
Exp/Cntr=0.3,0.1

Type RM Length L Ch R = 1 ,19575   ,902,902,902
BEGIN DESCRIPTION:
SHOCKLEY CREEK 18.0
END DESCRIPTION:
XS GIS Cut Line= 3
      2355675.01     13619824.97        2355825.       13619175.
      2355025.01     13618375.01
#Sta/Elev= 30
  4333.3  339.57  4406.8   337.9    4518  334.94  4618.9     333  4630.9  333.64
  4651.4   332.4  4682.2   332.6  4721.8   331.2  4764.3  330.43  4795.1  329.18
  4815.6  327.35  4848.1  326.54  4890.9   327.5  4990.1  327.34    5024  325.48
  5024.5  324.98  5033.2  325.48  5042.8  326.69  5141.8  328.48  5170.1  331.06
  5195.6  331.36  5240.8   332.5    5269  330.59  5311.5  332.04  5436.7  332.77
  5519.1  333.51    5695  334.34  5771.6   334.9  5976.2  336.01  6131.7  338.62
#Mann= 10 ,-1 , 0
  4333.3     .05       0  4406.8     .07       0  4721.8      .1       0
    5024     .05       0  5033.2      .1       0  5195.6     .07       0
  5436.7    .035       0  5519.1     .07       0    5695    .035       0
  5771.6     .05       0
Bank Sta=5024,5033.2
XS Rating Curve= 0 ,0
Exp/Cntr=0.3,0.1

Type RM Length L Ch R = 1 ,18673   ,466,466,466
BEGIN DESCRIPTION:
SHOCKLEY CREEK 17.0
END DESCRIPTION:
XS GIS Cut Line= 3
        2356225.     13619874.96        2356175.       13619225.
      2355774.99     13618324.97
#Sta/Elev= 30
  4351.7  335.99    4696  330.66  4722.8  329.94  4742.8  325.91  4752.8  321.02
  4762.9  322.28  4772.9  322.01  4778.3  320.43  4778.8  319.93  4787.5  320.43
    4793  322.93    4803  322.62    4813  324.91  4833.1   325.1  4853.1  321.69
  4863.2  325.13  4903.3  325.52  4953.4  323.83  4993.5  324.02  5006.3  322.69
  5012.5   320.5  5017.9  321.66  5025.5  327.14  5035.7   329.8  5063.4  330.32
  5116.4  332.05    5437  329.83  5601.7  332.73  5659.9  333.83  5988.5  335.54
#Mann= 8 ,-1 , 0
  4351.7     .07       0    4696      .1       0  4778.3     .05       0
  4787.5      .1       0  5063.4     .07       0    5437    .035       0
  5601.7     .05       0  5659.9    .035       0
Bank Sta=4778.3,4787.5
XS Rating Curve= 0 ,0
Exp/Cntr=0.3,0.1

Type RM Length L Ch R = 1 ,18207   ,909,909,909
BEGIN DESCRIPTION:
SHOCKLEY CREEK 16.0
END DESCRIPTION:
XS GIS Cut Line= 3
        2356425.       13620025.        2356625.       13619275.
      2355925.01     13618475.01
#Sta/Elev= 30
  4223.8  339.37  4368.7  334.56  4551.7  330.74  4696.4  329.13    4759  328.66
  4813.7  328.32  4857.9  324.96  4907.5  323.67  4958.6  325.15  4989.7  323.45
  4992.8  319.79  4993.3  319.29    5002  319.79  5013.8  320.54  5021.4  323.99
  5035.6  324.91  5099.2  325.63  5141.9  328.01  5240.6  330.76  5297.6   330.4
    5326  328.49  5377.8  327.46  5432.3  325.57  5567.1  325.82    5680  328.25
  5744.1  328.17  5860.3  332.25  5889.1  333.26  6004.9   334.6    6063  334.72
#Mann= 10 ,-1 , 0
  4223.8     .07       0  4696.4      .1       0    4759     .07       0
  4857.9      .1       0  4992.8     .05       0    5002      .1       0
  5377.8     .07       0  5860.3     .05       0  5889.1     .07       0
  6004.9    .035       0
Bank Sta=4992.8,5002
XS Rating Curve= 0 ,0
Exp/Cntr=0.3,0.1

Type RM Length L Ch R = 1 ,17298   ,1440,1440,1440
BEGIN DESCRIPTION:
SHOCKLEY CREEK 15.0
END DESCRIPTION:
XS GIS Cut Line= 3
      2356474.97     13620125.04        2357175.       13619125.
      2357425.02     13618574.96
#Sta/Elev= 30
  3779.2  341.64  4001.1  335.95  4030.8  333.85  4131.9  332.02  4152.9  330.64
  4295.8  328.17  4374.2  328.05  4453.7  327.51  4504.2  325.24  4573.7  323.61
  4605.4  323.21    4683  326.18  4719.2   324.9  4935.8  323.88  4950.6  323.59
  4963.3  322.09  4977.7  322.03  4985.2  317.84  4985.7  317.34  4999.8  317.84
  5021.9   318.6  5031.8  320.55  5054.8  322.11  5065.8  325.03  5083.4  325.45
  5088.9  326.34  5158.1  328.76  5206.3  329.17  5442.2  334.45  5604.1  338.91
#Mann= 7 ,-1 , 0
  3779.2     .07       0  4374.2     .12       0  4573.7      .1       0
  4985.2     .05       0  4999.8      .1       0  5206.3     .05       0
  5442.2     .07       0
Bank Sta=4985.2,4999.8
XS Rating Curve= 0 ,0
Exp/Cntr=0.3,0.1

Type RM Length L Ch R = 1 ,15858   ,887,887,887
BEGIN DESCRIPTION:
SHOCKLEY CREEK 14.0
END DESCRIPTION:
XS GIS Cut Line= 3
        2356875.       13620725.        2357775.       13619725.
        2357575.     13618525.02
#Sta/Elev= 30
  3654.1  342.97  3816.2  339.98  4170.9  331.04  4227.8  328.64  4248.7  326.13
  4284.6  326.88  4348.1  323.95    4369  326.37  4404.9  326.05  4425.8  328.45
  4496.8  328.56  4617.2  325.02  4674.9  320.72  4815.2  320.39  4900.4  321.86
    4964  319.97  4984.9  317.88  4985.4  317.38  4999.8  317.88  5027.3  322.13
    5040  321.66  5060.3  324.69  5112.4  325.32    5182  324.48  5311.4  326.71
  5624.2  328.46  5786.8  330.48  5901.9  332.66  5987.6  334.57    6216  340.87
#Mann= 11 ,-1 , 0
  3654.1     .05       0  3816.2     .07       0  4674.9      .1       0
  4984.9     .05       0  4999.8      .1       0  5112.4     .07       0
  5311.4    .035       0  5624.2     .05       0  5786.8    .035       0
  5901.9     .07       0  5987.6    .035       0
Bank Sta=4984.9,4999.8
XS Rating Curve= 0 ,0
Exp/Cntr=0.3,0.1

Type RM Length L Ch R = 1 ,14971   ,777,777,777
BEGIN DESCRIPTION:
SHOCKLEY CREEK 13.0
END DESCRIPTION:
XS GIS Cut Line= 3
      2357725.03     13620924.96        2358325.       13620225.
      2358870.16     13619142.09
#Sta/Elev= 30
  4073.7  338.91  4123.6  337.57  4152.1  337.98  4271.8  332.42  4392.5  330.11
  4428.7  328.25  4492.4  327.19  4513.2  328.05  4619.7  324.62  4654.8  325.41
  4683.3  324.16  4740.4   324.3  4783.2  322.61  4804.1  323.34  4872.9  322.56
  4896.3  320.96  4939.1  321.45  4981.9  319.91  5040.4  320.44    5069  319.65
  5069.5  319.15    5084  319.65  5143.5  320.55  5353.9  320.33    5428  321.66
  5612.1  320.93    5679  321.97  5782.4  326.38  6114.1     340    6208  340.92
#Mann= 5 ,-1 , 0
  4073.7     .07       0  4872.9      .1       0    5069     .05       0
    5084      .1       0  5782.4     .07       0
Bank Sta=5069,5084
XS Rating Curve= 0 ,0
Exp/Cntr=0.3,0.1

Type RM Length L Ch R = 1 ,14194   ,613,613,613
BEGIN DESCRIPTION:
E20827
END DESCRIPTION:
XS GIS Cut Line= 3
      2357721.57     13621244.99      2358653.15     13620662.04
      2359367.55      13619073.2
#Sta/Elev= 30
  3257.4  342.74  3455.7  337.22  3485.6  337.85  3528.8  335.97    3580  335.84
  3759.7  331.05  3869.5  328.95  3890.7  329.66  3911.4  328.24  4089.1   327.4
    4189  326.23    4217  327.09  4243.5  325.63  4561.4  323.11  4627.7  320.47
  4688.8  320.03  4717.4  322.51  4740.6  322.85  4780.7  321.62  4824.6  318.36
  4923.2  319.83  4983.1  318.77  4991.5  314.95    4992  314.45  5008.5  314.95
  5011.7  318.92    5203  321.86  5612.6  328.97  5710.7  333.07  6098.4  342.71
#Mann= 9 ,-1 , 0
  3257.4     .07       0  3759.7    .035       0  3911.4     .07       0
  4089.1    .035       0  4243.5     .07       0  4627.7      .1       0
  4991.5     .05       0  5008.5      .1       0    5203     .07       0
Bank Sta=4991.5,5008.5
XS Rating Curve= 0 ,0
Exp/Cntr=0.3,0.1

Type RM Length L Ch R = 1 ,13581   ,914,914,914
BEGIN DESCRIPTION:
SHOCKLEY CREEK 12.0
END DESCRIPTION:
XS GIS Cut Line= 3
      2357625.01     13621474.99        2359425.       13620275.
        2359825.       13619375.
#Sta/Elev= 30
  2840.8  348.51  3085.7  342.59  3172.8  339.07  3615.8  329.48  3820.2   327.9
  4204.4  324.01    4247  324.45    4309  321.78  4315.7  320.39  4339.1  314.74
  4339.6  314.24  4356.1  314.74  4413.7  317.66  4548.9  318.04  4636.1  315.83
  4679.6  317.64  4751.7  317.14  4888.4  319.71  4981.6  317.98  4996.6   315.4
  5018.5  318.93  5058.8  318.78    5104  322.03  5210.4  323.97  5339.8  327.72
  5529.7  331.01    5599  331.91  5770.1  338.81  5858.3  344.37    5989  350.21
#Mann= 14 ,-1 , 0
  2840.8     .07       0  3615.8    .035       0  3820.2     .07       0
  4204.4     .12       0    4309     .07       0  4315.7      .1       0
  4339.1     .05       0  4356.1      .1       0    5104     .07       0
  5210.4      .1       0  5339.8    .035       0  5529.7     .07       0
    5599    .035       0  5858.3     .07       0
Bank Sta=4339.1,4356.1
XS Rating Curve= 0 ,0
Exp/Cntr=0.3,0.1

Type RM Length L Ch R = 1 ,12667   ,428,428,428
BEGIN DESCRIPTION:
SHOCKLEY CREEK 11.0
END DESCRIPTION:
XS GIS Cut Line= 3
      2358974.98     13621775.04        2359775.       13620575.
        2359875.     13619375.02
#Sta/Elev= 30
    3566  342.21  3696.7  340.49  3830.2  335.29  3948.9  328.71  4015.7  326.41
  4181.2  324.53  4201.2  324.23  4572.1  320.29  4589.1  320.58  4647.7  317.61
  4964.7  317.03  4972.2  316.45  4978.2  314.18  4985.7  316.31  4985.8  311.79
  4986.3  311.29  5003.6  311.79  5010.8  312.16  5018.3   317.6  5038.4  320.45
  5076.5  321.75  5193.6  321.03  5306.5  321.38  5390.9  322.05  5489.5  323.21
  5660.5  326.47  5881.3  334.37  5931.5  336.37  6051.9   344.1  6212.4  350.59
#Mann= 14 ,-1 , 0
    3566     .05       0  3830.2    .035       0  3948.9     .07       0
  4015.7    .035       0  4181.2     .12       0  4201.2    .035       0
  4572.1      .1       0  4985.8     .05       0  5003.6      .1       0
  5076.5     .07       0  5193.6     .12       0  5306.5     .07       0
  5390.9     .12       0  5489.5     .07       0
Bank Sta=4985.8,5003.6
XS Rating Curve= 0 ,0
Exp/Cntr=0.3,0.1

Type RM Length L Ch R = 1 ,12239   ,464,464,464
BEGIN DESCRIPTION:
SHOCKLEY CREEK 10.0
END DESCRIPTION:
XS GIS Cut Line= 3
        2359025.       13621775.        2360025.       13620875.
        2360825.       13619775.
#Sta/Elev= 30
  3659.6  341.99  3784.1  338.98    3808  337.31  3829.6  333.15  3864.8  332.53
  3872.2  330.09  3886.4  332.12  3893.2  330.82  3900.6  334.13  3920.1  334.87
  4105.4  328.14  4410.4  321.85  4556.9   321.1  4686.2  316.56  4905.9  314.53
  4983.7  316.48  5001.6  311.93    5018  311.73  5018.5  311.23  5035.9  311.73
  5062.5  316.14    5163   316.7  5234.1  319.94    5559  321.67  5702.9  324.54
  5706.9  324.54  5814.4  326.05  6200.9  337.19  6292.8  341.66  6365.1  342.36
#Mann= 10 ,-1 , 0
  3659.6     .05       0  3784.1    .035       0  3920.1     .07       0
  4556.9      .1       0    5018     .05       0  5035.9      .1       0
    5559     .12       0  5702.9     .07       0  5706.9     .12       0
  5814.4     .07       0
Bank Sta=5018,5035.9
XS Rating Curve= 0 ,0
Exp/Cntr=0.3,0.1

Type RM Length L Ch R = 1 ,11775   ,478,478,478
BEGIN DESCRIPTION:
SHOCKLEY CREEK 9.0
END DESCRIPTION:
XS GIS Cut Line= 3
      2359825.02     13622174.96        2360425.       13620975.
      2360824.99     13619975.03
#Sta/Elev= 30
  3658.3  338.08  3677.6  337.63  3788.9  334.87  4078.2  327.85  4320.7  324.24
  4387.8  321.94  4404.5  322.49  4410.1  321.61  4583.4  321.18  4737.7  318.73
  4829.4  316.87  4865.7  317.43  4932.8  315.11  4963.6  315.41  4991.5  312.94
  5009.3  314.08  5012.4  312.44  5012.9  311.94  5030.4  312.44  5038.9  314.17
    5117  316.46  5139.9   318.4  5452.3  322.36  5497.8  321.89  5549.5  322.04
  5624.6  323.52  5660.9  325.92  5721.5  327.33    5906  334.56  6076.9  338.85
#Mann= 9 ,-1 , 0
  3658.3    .035       0  3677.6     .07       0  3788.9    .035       0
  4078.2     .07       0  4737.7      .1       0  5012.4     .05       0
  5030.4      .1       0  5497.8     .12       0  5549.5     .07       0
Bank Sta=5012.4,5030.4
XS Rating Curve= 0 ,0
Exp/Cntr=0.3,0.1

Type RM Length L Ch R = 1 ,11297   ,431,431,431
BEGIN DESCRIPTION:
SHOCKLEY CREEK 8.0
END DESCRIPTION:
XS GIS Cut Line= 3
      2360225.02     13622374.96        2360825.       13621175.
      2361525.03     13620174.96
#Sta/Elev= 30
  3663.8  338.06  3873.4  332.59  3918.1  332.35  3940.5   330.7  4018.5  328.99
  4127.4  326.59  4413.1  320.97  4437.6  320.85  4616.9  318.97    4670  320.29
    4730  316.88  4795.8  313.38  4885.2  314.89  4938.3   313.6  4960.7  314.52
  4965.6   310.4  4966.1   309.9  4983.7   310.4  5008.4  312.68  5012.8   314.2
  5033.7  315.15  5054.7  314.24  5129.5  316.72  5191.5  316.76  5221.2  317.97
  5328.4  316.98  5608.3  321.25  5974.5  333.24  6132.3  339.58  6226.1  341.33
#Mann= 9 ,-1 , 0
  3663.8     .07       0  4018.5    .035       0  4127.4     .07       0
  4413.1    .035       0  4437.6     .07       0    4730      .1       0
  4965.6     .05       0  4983.7      .1       0  5129.5     .07       0
Bank Sta=4965.6,4983.7
XS Rating Curve= 0 ,0
Exp/Cntr=0.3,0.1

Type RM Length L Ch R = 1 ,10866   ,453,453,453
BEGIN DESCRIPTION:
SHOCKLEY CREEK 7.0
END DESCRIPTION:
XS GIS Cut Line= 3
      2360625.02     13622174.97        2361025.       13621475.
        2361525.     13620274.99
#Sta/Elev= 30
  4187.6  331.15  4268.2  329.84  4319.3  327.85  4335.1  328.25  4348.8  327.06
  4399.9  326.47  4429.4  324.88  4443.1  325.47  4458.9  323.12  4523.7  322.63
  4553.8  321.53  4813.3  317.02  4958.5  315.01  4980.1  313.21    5003  313.08
  5006.4  310.79  5006.9  310.29  5024.5  310.79  5026.3  312.17  5037.7  313.23
  5061.5  312.77  5102.1  314.19  5138.4  313.41  5156.3  315.24  5191.5  316.54
    5289  315.14  5711.5   318.8    5828  322.48  6226.1  339.01  6293.8  340.85
#Mann= 6 ,-1 , 0
  4187.6     .07       0  4553.8    .035       0  4813.3     .07       0
  5006.4     .05       0  5024.5     .07       0    5289     .07       0
Bank Sta=5006.4,5024.5
XS Rating Curve= 0 ,0
Exp/Cntr=0.3,0.1

Type RM Length L Ch R = 1 ,10413   ,460,460,460
BEGIN DESCRIPTION:
SHOCKLEY CREEK 6.0
END DESCRIPTION:
XS GIS Cut Line= 3
      2360725.02     13622174.98        2361425.       13621475.
      2361624.99     13620375.05
#Sta/Elev= 30
  4015.1  330.55  4057.5  329.97  4142.3  326.85  4198.9  326.07  4376.1  321.41
  4399.3  321.04  4484.3  319.37  4683.9  316.26  4788.2     315  4863.6  313.96
  4948.4  313.81  4976.7  312.07  4990.9  310.88  4992.4  310.18  4992.9  309.68
    5010  309.68  5010.5  310.18  5015.2  311.52  5055.8  314.75  5119.7  316.05
  5228.6  314.52  5359.2  316.06  5513.2  317.42  5649.2   320.3  5755.9  324.19
  5767.3  325.25  5926.1  332.09  5990.9  334.07  6037.9  336.75    6123  338.94
#Mann= 10 ,-1 , 0
  4015.1     .07       0  4376.1    .035       0  4399.3     .07       0
  4484.3    .035       0  4683.9     .07       0  4788.2      .1       0
  4992.4     .05       0  5010.5      .1       0  5119.7    .035       0
  5359.2     .07       0
Bank Sta=4992.4,5010.5
XS Rating Curve= 0 ,0
Exp/Cntr=0.3,0.1

Type RM Length L Ch R = 1 ,9953    ,309,309,309
BEGIN DESCRIPTION:
SHOCKLEY CREEK 5.0
END DESCRIPTION:
XS GIS Cut Line= 3
      2360875.01     13622224.99        2361775.       13621725.
        2361675.     13620525.01
#Sta/Elev= 30
  3970.1  329.74  4008.9  328.74  4037.6  328.97    4073  327.66    4207  325.45
  4233.2  324.62  4308.7  324.64  4389.9  322.86    4419  321.52  4430.3  321.37
  4595.8  317.67  4667.9  316.67  4677.1  317.17  4726.2  315.34  4844.7  313.93
  4850.9  313.32  4964.2   313.5  4976.9  308.38  4977.4  307.88    4995  308.38
  4996.8  309.42  5009.7  309.68  5029.8  313.74  5120.1  314.59    5293  315.84
  5360.9   315.5  5422.3  314.11    5544  314.56  5664.4  316.74  6203.8  333.54
#Mann= 11 ,-1 , 0
  3970.1     .07       0  4008.9     .05       0    4207     .07       0
    4419    .035       0  4430.3     .07       0  4844.7      .1       0
  4976.9     .05       0    4995      .1       0  5120.1     .07       0
    5293    .035       0  5422.3     .07       0
Bank Sta=4976.9,4995
XS Rating Curve= 0 ,0
Exp/Cntr=0.3,0.1

Type RM Length L Ch R = 1 ,9644    ,568,568,568
BEGIN DESCRIPTION:
E20826
END DESCRIPTION:
XS GIS Cut Line= 4
      2360722.14     13622811.01      2361950.92     13622028.01
      2362145.25     13621622.22      2362951.13     13620827.77
#Sta/Elev= 30
  3373.8  332.73  3673.8  329.61  3740.5  329.26  3815.9  326.35  3940.6  325.41
  4155.6  323.41  4213.1  320.81  4510.2  320.09  4561.8  317.43  4574.8  319.31
  4947.5  315.06  4978.3  313.58  4987.3   308.1  4991.4  308.04  4991.9  307.54
  5009.6  308.04    5010  310.81  5022.7  312.14  5050.2  312.27  5111.7  312.71
  5134.4  310.11  5202.4  313.46    5314  312.24  5422.8  314.55  5497.8  316.46
  5600.4  314.71  5756.7  315.96  5873.4  317.57  5922.7  318.38  6412.4  334.44
#Mann= 12 ,-1 , 0
  3373.8     .05       0  3673.8     .07       0  3740.5     .05       0
  3940.6     .07       0  4991.4     .05       0  5009.6     .07       0
  5050.2      .1       0  5422.8     .07       0  5600.4     .12       0
  5756.7     .07       0  5873.4     .12       0  5922.7     .07       0
Bank Sta=4991.4,5009.6
XS Rating Curve= 0 ,0
Exp/Cntr=0.3,0.1

Type RM Length L Ch R = 1 ,9076    ,455,455,455
BEGIN DESCRIPTION:
SHOCKLEY CREEK 4.0
END DESCRIPTION:
XS GIS Cut Line= 3
      2360725.01       13623125.        2362525.       13621775.
      2363725.02     13620674.98
#Sta/Elev= 30
  2744.8  338.22  2786.1  338.04  2967.5   335.6  3094.2   332.9  3219.9  329.73
  3650.1  323.23  4072.9   320.7  4552.1  311.11  4644.8  315.22  4814.6   313.1
  4872.9  313.04  4894.8   309.9  4912.1  313.06  4981.3  312.31  4998.2  310.03
  4999.2  307.19  4999.7  306.69  5018.1  307.19  5029.5  310.22  5044.4  312.61
  5130.1  313.94  5678.2  324.18  5808.7  325.18  5879.3  330.09  5963.1  331.87
  5978.6  330.73  6204.9  341.51  6233.3   339.6  6261.6  343.65  6622.7  358.94
#Mann= 14 ,-1 , 0
  2744.8     .12       0  2786.1     .07       0  2967.5     .12       0
  3094.2     .07       0  3219.9     .05       0  3650.1     .07       0
  4814.6      .1       0  4912.1     .07       0  4999.2     .05       0
  5018.1     .07       0  5029.5      .1       0  5130.1     .07       0
  5678.2     .12       0  5963.1     .07       0
Bank Sta=4999.2,5018.1
XS Rating Curve= 0 ,0
Exp/Cntr=0.3,0.1

Type RM Length L Ch R = 1 ,8621    ,443,443,443
BEGIN DESCRIPTION:
SHOCKLEY CREEK 3.0
END DESCRIPTION:
XS GIS Cut Line= 3
      2360824.97     13623175.02        2362625.       13622125.
      2363224.97     13621575.03
#Sta/Elev= 30
    2924  340.25  2981.9  339.25  3047.4  338.15  3291.9  332.22  3294.5  332.11
  3765.4  323.39  4035.4   320.8    4102  320.73  4107.8  321.99  4189.7  320.29
  4452.2  315.62  4510.1  313.45    4556  313.86    4685  311.09  4896.2  311.72
  5011.3  311.24    5015  306.51  5021.8  307.58  5026.5  306.48    5027  305.98
  5045.5  306.48  5050.1  310.09  5057.5  312.36  5071.7   312.8  5184.6   312.4
  5234.5  309.73  5248.7  311.94  5374.5  315.34  5637.8  322.83  5821.8  331.62
#Mann= 10 ,-1 , 0
    2924     .12       0  2981.9     .07       0  3047.4     .12       0
  3291.9     .07       0  3294.5     .05       0  4189.7     .07       0
  4896.2      .1       0  5026.5     .05       0  5045.5      .1       0
  5374.5     .07       0
Bank Sta=5026.5,5045.5
XS Rating Curve= 0 ,0
Exp/Cntr=0.3,0.1

Type RM Length L Ch R = 1 ,8178    ,1304,1304,1304
BEGIN DESCRIPTION:
SHOCKLEY CREEK 2.0
END DESCRIPTION:
XS GIS Cut Line= 3
      2361375.01       13622925.        2362575.       13622525.
        2363775.       13621625.
#Sta/Elev= 30
  3739.7  327.61  4055.9  322.26  4400.4   319.4  4545.1  317.87  4841.2  314.07
  4925.5  311.82  4951.9  310.19    4973  310.58  4984.6  309.22  4985.1  308.72
  5003.6  309.22  5004.6  310.75  5032.7  311.92  5091.1  310.66  5244.8  313.24
  5426.5  312.83  5511.9  311.22  5518.1  309.68  5526.5  309.24  5545.4  311.13
  5568.1  310.44  5641.1  311.11  5685.6  312.53  5926.5  319.09  6011.9     323
  6041.1  326.13  6111.9  329.15  6141.1  332.07  6391.1  346.03  6504.6   349.5
#Mann= 9 ,-1 , 0
  3739.7     .05       0  4400.4     .07       0  4545.1     .12       0
  4841.2      .1       0  4984.6     .05       0  5003.6      .1       0
  5244.8     .07       0  5545.4      .1       0  5685.6     .07       0
Bank Sta=4984.6,5003.6
XS Rating Curve= 0 ,0
Exp/Cntr=0.3,0.1

Type RM Length L Ch R = 1 ,6874    ,233,233,233
BEGIN DESCRIPTION:
SHOCKLEY CREEK 1.0
END DESCRIPTION:
XS GIS Cut Line= 3
      2361175.01       13623075.        2363575.       13622675.
      2364174.97     13622125.02
#Sta/Elev= 30
  2579.4  333.29  2703.5  330.95  3045.7  323.67  3438.7  319.63  3795.9  317.53
  3986.2  314.54  4022.8  314.09  4100.1  311.07  4150.9  313.36  4370.6  312.54
  4576.6  312.16  4637.4  310.82  4748.9  312.45    4876   309.2  4961.8  308.44
  4969.8  305.37  4970.3  304.87  4989.2  305.37  4992.2  306.83  5019.6  308.37
  5430.3  316.37  5559.6  322.29  5621.4  326.28  5649.8  326.19  5684.9  328.22
  5691.7  329.75  5713.3  329.97  5727.5  332.18  5762.6  332.79  5826.4  337.28
#Mann= 11 ,-1 , 0
  2579.4     .07       0  2703.5     .05       0  3438.7     .07       0
  3986.2      .1       0  4022.8     .07       0  4150.9      .1       0
  4370.6     .07       0    4876      .1       0  4969.8     .05       0
  4989.2      .1       0  5559.6     .07       0
Bank Sta=4969.8,4989.2
XS Rating Curve= 0 ,0
Exp/Cntr=0.3,0.1

Type RM Length L Ch R = 1 ,6641    ,292,292,292
BEGIN DESCRIPTION:
E20825
END DESCRIPTION:
XS GIS Cut Line= 4
       2362305.3     13623411.13      2363579.81     13622953.91
      2363877.01     13622696.71      2364378.91     13622229.04
#Sta/Elev= 30
  3514.6  318.25  3535.6  317.93  3779.5  316.72  3810.3  314.95  3815.6  315.85
  3822.4  314.38  3854.3   316.1    3964   315.7  4629.8  310.54    4706  311.14
  4731.4  309.87  4778.5  311.28  4963.9  311.36  5006.6  310.24  5011.2  304.15
  5011.7  303.65  5030.6  304.15  5034.2  306.77  5041.8  307.84  5087.9  309.43
  5148.1  307.48  5211.8  309.58  5367.8  310.84  5635.4  321.39  5664.9  325.01
  5671.7  323.55    5679  324.95  5693.2  324.51  5721.5  329.92  5947.7  342.88
#Mann= 6 ,-1 , 0
  3514.6     .05       0  3535.6     .07       0  5011.2     .05       0
  5030.6     .07       0  5087.9      .1       0  5635.4     .07       0
Bank Sta=5011.2,5030.6
XS Rating Curve= 0 ,0
Exp/Cntr=0.3,0.1

Type RM Length L Ch R = 1 ,6349    ,277,277,277
BEGIN DESCRIPTION:
E20824
END DESCRIPTION:
XS GIS Cut Line= 4
      2362693.94     13623656.89      2363825.57     13623056.78
      2364054.19     13622879.61      2364362.81     13622485.26
#Sta/Elev= 30
  3595.9  317.62  3694.7  315.87  3930.3  314.59  4381.4  311.59  4469.4  312.11
    4612  308.89  4743.9  310.79  4782.3  308.06  4787.9  309.51  4831.9  310.55
  4898.4   310.3  4941.3  310.35  4970.2  309.03  4981.4  304.41  4981.9  303.91
  5000.8  304.41  5005.5   307.4  5034.5  308.76  5098.8  307.51  5134.1  307.98
  5148.6  307.08  5319.7  309.13  5334.2  310.65  5340.5  313.21  5419.2  316.19
  5504.2  320.95  5533.6  321.46    5647  325.82  5661.5  328.12  5666.8  326.78
#Mann= 6 ,-1 , 0
  3595.9     .05       0  3930.3     .07       0  4898.4      .1       0
  4981.4     .05       0  5000.8      .1       0  5533.6     .07       0
Bank Sta=4981.4,5000.8
XS Rating Curve= 0 ,0
Exp/Cntr=0.3,0.1

Type RM Length L Ch R = 1 ,6072    ,206,206,206
BEGIN DESCRIPTION:
E20823
END DESCRIPTION:
XS GIS Cut Line= 3
      2362911.12     13623776.92      2364008.46      13623285.4
      2364385.69      13622622.4
#Sta/Elev= 30
  3670.7   315.4    3766  314.35  3986.4  313.57  4091.3  314.65  4123.3  311.25
  4157.5  312.22  4312.5  311.02  4539.5  310.81  4573.6  309.47  4666.4   308.7
  4759.1  310.35  4915.2  311.41  4924.8  310.59  4942.6  308.35  4980.1     308
    4992  304.02  4992.5  303.52  5011.4  304.02  5017.6  306.32  5023.3  305.71
  5039.2  306.77  5046.1  308.22  5098.3  308.11  5157.4  310.31  5275.6  310.77
  5297.2  311.97  5323.5  311.51  5405.3  313.53  5560.9  320.19  5635.9  322.29
#Mann= 8 ,-1 , 0
  3670.7     .05       0    3766     .07       0  3986.4     .05       0
  4312.5     .07       0  4924.8      .1       0    4992     .05       0
  5011.4      .1       0  5323.5    .035       0
Bank Sta=4992,5011.4
XS Rating Curve= 0 ,0
Exp/Cntr=0.3,0.1

Type RM Length L Ch R = 1 ,5866    ,240,240,240
BEGIN DESCRIPTION:
E20822
END DESCRIPTION:
XS GIS Cut Line= 3
      2363014.01     13623902.65       2364134.2       13623434.
      2364597.15     13622725.29
#Sta/Elev= 30
  3568.8  314.33  3668.3  313.48  3765.9  312.54  3877.2  313.18  3932.1  312.59
  4296.8  309.35  4437.1  309.81  4469.6  307.45  4502.1  309.53  4620.7  309.57
  4689.6  309.54  4728.7  309.41  4876.5  309.79  4968.8  306.22  4984.9  305.28
  4998.3  301.45  4998.8  300.95  5017.7  301.45  5020.8  305.26    5035  306.38
  5199.8  309.13  5246.3  309.81  5273.3  312.25  5315.2     312  5433.2  317.48
  5547.8  322.78    5563  324.83  5570.2  328.21  5593.2  323.46  5629.6  325.11
#Mann= 16 ,-1 , 0
  3568.8     .05       0  3668.3     .07       0  3765.9     .05       0
  3877.2     .07       0  3932.1     .05       0  4296.8     .07       0
  4620.7    .035       0  4689.6     .07       0  4728.7    .035       0
  4876.5     .07       0  4968.8      .1       0  4998.3     .05       0
  5017.7      .1       0  5199.8     .05       0  5315.2    .035       0
  5433.2     .07       0
Bank Sta=4998.3,5017.7
XS Rating Curve= 0 ,0
Exp/Cntr=0.3,0.1

Type RM Length L Ch R = 1 ,5626    ,401,401,401
BEGIN DESCRIPTION:
E20821
END DESCRIPTION:
XS GIS Cut Line= 3
       2363031.1     13623994.12      2364259.94     13623565.45
       2364991.5     13622828.18
#Sta/Elev= 30
    3430  314.14  3689.5  312.22  3794.2  313.14  4118.7  308.88  4329.2  309.03
  4429.3  309.59  4434.5  309.52  4501.8  308.22  4539.8   308.8  4841.4  309.26
  4890.9  306.05  4926.3  306.58    4952  305.23  4975.8  307.15  5004.1  304.23
  5008.5  299.42    5009  298.92  5027.9  299.42  5046.5  303.08  5053.6  306.41
  5103.1   306.5  5123.4   308.3  5138.4  310.03    5166  310.63  5356.4  313.56
  5456.6  316.89  5463.7  318.75  5477.9  319.66  5511.7  319.62  5770.1   327.3
#Mann= 13 ,-1 , 0
    3430     .05       0  4118.7     .07       0  4329.2    .035       0
  4429.3     .07       0  4434.5    .035       0  4539.8     .07       0
    4952      .1       0  5008.5     .05       0  5027.9      .1       0
  5123.4     .07       0    5166     .05       0  5356.4    .035       0
  5511.7     .05       0
Bank Sta=5008.5,5027.9
XS Rating Curve= 0 ,0
Exp/Cntr=0.3,0.1

Type RM Length L Ch R = 1 ,5225    ,545,545,545
BEGIN DESCRIPTION:
E20820
END DESCRIPTION:
XS GIS Cut Line= 3
      2363014.02     13624154.13      2364597.15     13623702.62
      2365321.49     13623086.65
#Sta/Elev= 30
  3101.1  315.43  3257.9  312.84  3675.2  311.01    3789  309.77  3995.4  309.96
  4266.8  307.53  4394.5  309.33  4462.2  308.98  4568.3  307.51  4607.9  305.73
  4672.3  306.77  4713.9  305.19  4800.7  306.31  4857.8  308.43  4970.9  304.23
  5013.7  306.75    5028  305.53  5032.5  295.75    5033  295.25    5052  295.75
  5056.6  306.47  5070.5  306.79  5217.6   309.2  5364.6  312.56  5371.3   312.7
  5503.6  314.29  5511.7  315.71  5636.1  317.89  5688.1  319.42  5698.2  321.21
#Mann= 14 ,-1 , 0
  3101.1     .05       0  3257.9     .07       0  3675.2     .05       0
    3789    .035       0  3995.4     .07       0  4672.3      .1       0
  5032.5     .05       0    5052      .1       0  5070.5     .07       0
  5217.6     .05       0  5364.6     .07       0  5371.3    .035       0
  5511.7     .05       0  5636.1     .07       0
Bank Sta=5032.5,5052
XS Rating Curve= 0 ,0
Exp/Cntr=0.3,0.1

Type RM Length L Ch R = 1 ,4680    ,639,639,639
BEGIN DESCRIPTION:
E20819
END DESCRIPTION:
XS GIS Cut Line= 4
      2363094.04     13624474.19      2364620.01     13624068.41
      2365162.97     13623616.89      2365550.83     13623092.14
#Sta/Elev= 30
    3245  313.18  3432.2  311.18  3711.6  311.38  4073.5  307.86  4332.5  308.66
  4424.6  307.01  4597.6  308.78  4767.1  307.83  4843.6   306.3  4939.2  307.14
  4993.3  306.39  4999.8  304.18  5004.4  295.49  5004.9  294.99  5023.9  295.49
  5042.8  305.79  5064.6  306.15  5107.5  304.14  5120.9   303.9  5163.9  306.93
  5213.3  308.29  5402.2   307.5  5571.4  308.06    5696  309.12  5761.6  309.91
  5876.5  313.21  5897.3  312.58  5941.2  315.15  6076.9  317.48  6182.7  321.68
#Mann= 9 ,-1 , 0
    3245     .05       0  4597.6     .07       0  4939.2     .12       0
  5004.4     .05       0  5023.9     .12       0  5107.5      .1       0
  5402.2     .07       0  5571.4      .1       0    5696     .07       0
Bank Sta=5004.4,5023.9
XS Rating Curve= 0 ,0
Exp/Cntr=0.3,0.1

Type RM Length L Ch R = 1 ,4041    ,1991,1991,1991
BEGIN DESCRIPTION:
E20818
END DESCRIPTION:
XS GIS Cut Line= 4
      2363042.57     13624554.21      2364808.62     13624428.48
       2365248.7     13624171.28       2365648.7     13623159.85
#Sta/Elev= 30
  2863.3     313  3146.4  310.89  3607.6  310.37  3888.3  306.96  4419.7  307.65
  4670.3  305.73  4797.5  306.81  4905.9  306.52    4948  306.86  4953.9     305
  4967.4  293.97  4967.9  293.47  4986.9  293.97    4991  298.79  5000.3   303.7
    5030  306.33  5178.2  307.21  5244.6  307.04  5376.1  306.34    5392  305.32
  5408.4  301.08  5421.8  300.41  5451.5  304.94  5487.6  306.16  5623.5  307.09
  5662.4  304.66  5746.2  304.36  5838.5  308.93    5899  309.54  6231.2  319.69
#Mann= 10 ,-1 , 0
  2863.3     .05       0  4797.5     .07       0  4905.9      .1       0
  4967.4     .05       0  4986.9      .1       0    5030     .07       0
  5178.2      .1       0  5244.6     .07       0  5487.6      .1       0
    5899     .07       0
Bank Sta=4967.4,4986.9
XS Rating Curve= 0 ,0
Exp/Cntr=0.3,0.1

Type RM Length L Ch R = 1 ,2050    ,0,0,0
BEGIN DESCRIPTION:
E20817
END DESCRIPTION:
XS GIS Cut Line= 4
      2363059.69     13624634.23      2364871.49     13624937.15
       2365843.1     13624451.34      2366608.38     13623269.16
#Sta/Elev= 30
    2256   313.1  2476.2  310.82  3153.6  306.53  3356.4  307.66  3853.2  307.37
  4339.6  305.53  4418.7  306.12  4601.7  304.75    4743     305  4852.2  305.26
  4946.6  305.31  4955.4  302.25    4959  291.61  4959.5  291.11  4978.9  291.61
  4983.3  297.62  4991.3  301.63  5005.7  303.26  5072.8  305.08  5258.3  303.75
  5329.7  304.37  5352.6  305.37  5358.5  306.47  5373.7  305.55  5393.5   306.4
  5525.4  304.73  5865.8  305.53  6065.9  307.46  6225.8  307.35  6587.5  309.58
#Mann= 10 ,-1 , 0
    2256     .05       0  4339.6     .07       0  4601.7     .12       0
    4743     .07       0  4852.2      .1       0    4959     .05       0
  4978.9      .1       0  5393.5     .07       0  5525.4     .12       0
  6065.9     .07       0
Bank Sta=4959,4978.9
XS Rating Curve= 0 ,0
Exp/Cntr=0.3,0.1

Chan Stop Cuts=-1
Use User Specified Reach Order=0
Composite Channel Slope=5
