--- Stream0755.prj (project) ---

Proj Title=Stream0755 Base Level Engineering
Current Plan=p01
Default Exp/Contr=0.3,0.1
English Units
Geom File=g01
Flow File=f01
Plan File=p01
Y Axis Title=Elevation
X Axis Title(PF)=Main Channel Distance
X Axis Title(XS)=Station
BEGIN DESCRIPTION:
Stream0755
END DESCRIPTION:
DSS Export Rating Curves= 0
DSS Export Rating Curve Sorted= 0
DSS Export Volume Flow Curves= 0
DXF OffsetX= 0
DXF OffsetY= 0
DXF ScaleX= 1
DXF ScaleY= 10

--- Stream0755.p01 (plan) ---

Plan Title=Multiple Run
Short Identifier=Multiple
Geom File=g01
Flow File=f01
Subcritical Flow
K Sum by GR= 0
Std Step Tol= 0.01
Critical Tol= 0.01
Num of Std Step Trials= 20
Max Error Tol= 0.3
Flow Tol Ratio= 0.001
Split Flow NTrial= 30
Split Flow Tol= 0.02
Split Flow Ratio= 0.02
Log Output Level= 0
Friction Slope Method= 1
Unsteady Friction Slope Method= 2
Unsteady Bridges Friction Slope Method= 1
Parabolic Critical Depth
Global Vel Dist=  1 , 1 , 1
Global Log Level= 0
CheckData=True
Encroach Param= -1, 0, 0, 0
BEGIN DESCRIPTION:
Multiple Run
END DESCRIPTION:

--- Stream0755.f01 (steady flow) ---

Flow Title=Multiple
Number of Profiles=7
Profile Names=10-year,25-year,50-year,1pct_min,100-year,1pct_plu,500-year
River Rch & RM= Stream0755,Reach-1,26099
     676    1085    1452     941    1878    3747    3110
River Rch & RM= Stream0755,Reach-1,23220
     892    1451    1960    1281    2555    5098    4301
River Rch & RM= Stream0755,Reach-1,17374
    1193    1966    2678    1762    3515    7013    6000
River Rch & RM= Stream0755,Reach-1,11479
    1354    2242    3063    2021    4032    8044    6919
River Rch & RM= Stream0755,Reach-1,6018
    1948    3274    4518    3006    5998   11969   10481
Boundary for River Rch & Prof#=Stream0755,Reach-1,1
Up Type=0
Dn Type=3
Dn Slope=0.005
Boundary for River Rch & Prof#=Stream0755,Reach-1,2
Up Type=0
Dn Type=3
Dn Slope=0.005
Boundary for River Rch & Prof#=Stream0755,Reach-1,3
Up Type=0
Dn Type=3
Dn Slope=0.005
Boundary for River Rch & Prof#=Stream0755,Reach-1,4
Up Type=0
Dn Type=3
Dn Slope=0.005
Boundary for River Rch & Prof#=Stream0755,Reach-1,5
Up Type=0
Dn Type=3
Dn Slope=0.005
Boundary for River Rch & Prof#=Stream0755,Reach-1,6
Up Type=0
Dn Type=3
Dn Slope=0.005
Boundary for River Rch & Prof#=Stream0755,Reach-1,7
Up Type=0
Dn Type=3
Dn Slope=0.005

--- Stream0755.g01 (geometry) ---

Geom Title=Existing Conditions
Program Version=4.10

River Reach=Stream0755      ,Reach-1
Reach XY= 30
        2469225.       13661925.      2468490.21     13661825.23
      2468021.31     13662067.35      2467745.18     13661574.56
      2467323.75     13662021.55      2466868.83     13661867.14
      2466028.45     13660723.75      2466119.66     13660022.26
      2465482.47      13659631.7      2465666.23      13659368.2
      2464932.67     13658831.53      2464792.14     13658141.03
      2463976.46     13658121.46      2463164.76     13657764.65
      2462964.72     13657375.98      2462476.43     13657721.99
      2461985.43     13657085.96      2461288.65     13656888.33
      2461282.79     13655021.57      2461673.51      13654730.9
        2460978.      13654423.6      2460871.88     13652825.99
      2460485.47     13652634.82      2460319.55     13651922.54
      2459975.52     13651714.55      2460322.77     13650480.93
      2459767.25     13649368.45      2459444.22     13649395.59
      2459519.55     13649022.53        2458925.       13648475.

Type RM Length L Ch R = 1 ,26099   ,600,600,600
BEGIN DESCRIPTION:
Stream0755 51.0
END DESCRIPTION:
XS GIS Cut Line= 3
      2469221.85      13661435.5      2469141.54     13661853.11
      2469021.07     13662479.57
#Sta/Elev= 30
  4413.3  307.52  4472.4  306.33  4616.5  301.24  4638.4  301.34  4690.4  297.72
  4708.1  297.98  4748.8  295.05  4797.2  293.58    4837  289.98  4851.3  289.59
  4860.9  290.84    4871  290.97  4898.1  289.67  4932.1  290.81  4983.1   290.6
  4993.2  290.22    5002  285.85  5007.1  287.62  5011.6  285.58  5011.9  285.08
  5015.4  285.08  5015.6  285.58  5023.8   291.1  5048.1   291.9  5110.9  293.93
  5147.9  294.44  5247.6  297.79  5349.4  302.22  5364.5  303.02  5476.5  307.55
#Mann= 9 ,-1 , 0
  4413.3     .07       0  4797.2      .1       0  5011.6     .05       0
  5015.6      .1       0  5048.1     .07       0  5147.9     .05       0
  5247.6     .07       0  5349.4     .05       0  5364.5     .07       0
Bank Sta=5011.6,5015.6
XS Rating Curve= 0 ,0
Exp/Cntr=0.3,0.1

Type RM Length L Ch R = 1 ,25499   ,473,473,473
BEGIN DESCRIPTION:
Stream0755 50.0
END DESCRIPTION:
XS GIS Cut Line= 3
        2468775.     13661574.98        2468675.       13661925.
        2468675.     13662224.98
#Sta/Elev= 30
  4643.7  297.98  4665.8  297.86  4758.1   293.6  4802.5  292.54  4830.9  291.45
  4851.7  291.58  4903.7  290.39  4912.8  290.83  4930.1  289.66  4951.8  287.73
    4957  288.22  4966.1  287.62  4997.3  287.93  5010.2  287.21  5015.7  283.49
    5016  282.99  5019.5  282.99  5019.8  283.49  5027.7  285.31  5037.7  288.39
  5097.7  285.05  5117.7  285.27  5127.7  286.41  5137.7  286.76  5156.3  289.42
  5207.7  293.75  5247.7  295.66  5267.7  297.75  5297.7  299.48  5307.7  299.59
#Mann= 6 ,-1 , 0
  4643.7     .12       0  4802.5     .07       0  4930.1      .1       0
  5015.7     .05       0  5019.8      .1       0  5156.3     .07       0
Bank Sta=5015.7,5019.8
XS Rating Curve= 0 ,0
Exp/Cntr=0.3,0.1

Type RM Length L Ch R = 1 ,25026   ,395,395,395
BEGIN DESCRIPTION:
E21320
END DESCRIPTION:
XS GIS Cut Line= 3
      2468488.54     13661348.82      2468323.38     13661887.37
      2468388.01     13662404.34
#Sta/Elev= 30
  4311.3  297.58  4336.9  296.32  4432.8   294.6  4544.4  290.94  4680.1  288.75
  4736.1  288.91  4757.1   287.9    4778  287.87  4783.5  288.66  4799.7  287.88
  4861.7   287.2  4870.8  286.18  4922.6  286.42  4932.8  285.51  4962.9  286.34
  4983.1  285.98  4993.1  284.63  5001.2   280.7  5001.4   280.2  5005.3   280.7
  5008.4   283.6  5013.5   285.1  5019.8  285.35  5033.5  285.88    5089  291.73
  5184.6  296.28  5255.3  301.17  5285.4  301.79  5325.7  304.23  5395.6  305.94
#Mann= 6 ,-1 , 0
  4311.3     .07       0  4544.4     .12       0  4799.7      .1       0
  5001.2     .05       0  5005.3      .1       0  5019.8     .07       0
Bank Sta=5001.2,5005.3
XS Rating Curve= 0 ,0
Exp/Cntr=0.3,0.1

Type RM Length L Ch R = 1 ,24631   ,351,351,351
BEGIN DESCRIPTION:
Stream0755 49.0
END DESCRIPTION:
XS GIS Cut Line= 3
      2468298.29     13661258.85        2468025.       13662075.
      2468129.65     13662495.58
#Sta/Elev= 30
  4147.4  295.13  4248.8  292.91  4322.6  292.41  4375.1  290.65    4407  290.95
  4486.3  288.88  4618.8  286.59  4645.1   287.4  4686.7  286.07  4723.4  284.04
  4739.8  285.83  4786.6  285.96  4818.3  282.92    4866  285.02  4871.3  284.28
  4960.7  284.59  4976.5  282.11    4985  278.74  4985.2  278.24  4989.1  278.74
  4992.3  282.71  4997.6  279.56  5005.5  283.25  5010.7  283.25  5017.6  285.01
  5090.5  289.19  5296.6  295.82  5356.7  295.76  5403.2  297.14  5441.5  295.85
#Mann= 8 ,-1 , 0
  4147.4     .07       0  4248.8     .12       0  4375.1     .07       0
  4486.3     .12       0  4686.7      .1       0    4985     .05       0
  4989.1      .1       0  5017.6     .07       0
Bank Sta=4985,4989.1
XS Rating Curve= 0 ,0
Exp/Cntr=0.3,0.1

Type RM Length L Ch R = 1 ,24280   ,539,539,539
BEGIN DESCRIPTION:
Stream0755 48.0
END DESCRIPTION:
XS GIS Cut Line= 3
      2468175.02     13661424.97      2467816.44     13661837.05
      2467525.01     13662474.98
#Sta/Elev= 30
  4467.8   291.4  4517.7  290.38  4538.6  290.88  4595.5  288.87  4638.3  288.97
  4659.2  287.67  4780.8  286.12    4851  284.77  4878.8   282.5  4886.1  280.56
  4892.7  280.12  4900.3  281.11    4907  280.37  4921.2  282.57  5006.7  282.57
  5020.7  277.15    5021  276.65  5024.8  277.15  5028.9  281.97  5034.4  282.73
    5098  281.47  5126.5  284.56  5201.1  284.37  5276.9   281.4  5367.8  280.85
  5396.6  282.85  5442.4  283.04  5603.6  289.81  5609.1  289.26  5715.4  291.81
#Mann= 5 ,-1 , 0
  4467.8     .12       0  4780.8      .1       0  5020.7     .05       0
  5024.8      .1       0  5276.9     .07       0
Bank Sta=5020.7,5024.8
XS Rating Curve= 0 ,0
Exp/Cntr=0.3,0.1

Type RM Length L Ch R = 1 ,23741   ,521,521,521
BEGIN DESCRIPTION:
Stream0755 47.0
END DESCRIPTION:
XS GIS Cut Line= 3
      2467607.64     13661170.47        2467575.       13661575.
        2467475.     13662375.03
#Sta/Elev= 30
  4589.6  289.94  4694.5  288.88  4824.9  289.09  4943.3   288.1  4955.3  287.96
  4985.4  282.81  4992.9  276.13    4998  276.13  5003.4  274.84  5003.7  274.34
  5007.6  274.84  5015.6  280.53  5038.3   280.2  5051.6  280.85  5086.1  279.31
  5106.3   279.3  5113.9  280.82  5118.9  279.13  5156.7  282.14  5166.8  281.41
  5186.9  282.81  5199.5  282.27  5275.1  282.85  5360.8  281.92  5408.6  279.11
  5469.1  279.05  5479.2  278.26  5544.4  280.45    5711  288.06  5801.7  290.19
#Mann= 6 ,-1 , 0
  4589.6     .07       0  4943.3     .12       0  5003.4     .05       0
  5007.6     .12       0  5051.6      .1       0  5544.4     .07       0
Bank Sta=5003.4,5007.6
XS Rating Curve= 0 ,0
Exp/Cntr=0.3,0.1

Type RM Length L Ch R = 1 ,23220   ,421,421,421
BEGIN DESCRIPTION:
E21319
END DESCRIPTION:
XS GIS Cut Line= 4
      2467562.21     13661449.39      2467504.79     13661564.24
      2467325.27      13661729.4      2467353.99     13662576.77
#Sta/Elev= 30
  4342.1   288.4  4422.7  287.54  4619.7   282.2  4766.9  281.19  4790.1  281.55
  4820.1  278.69  4870.1  279.02  4950.2  276.83  4960.2  277.66  4978.1  272.18
  4978.3  271.68  4982.4  272.18  4990.2  274.52  5000.2  273.63  5010.2   276.8
  5030.2  279.22  5130.3  278.88  5152.3  278.38  5166.1  276.55  5170.3  275.71
  5190.3  281.03  5220.3  284.75  5240.3  283.03  5270.4  282.84  5290.4  286.75
  5310.4  288.63  5340.4  289.07  5350.4   287.6  5380.4  291.06  5562.3   295.5
#Mann= 6 ,-1 , 0
  4342.1     .07       0  4422.7     .12       0  4766.9      .1       0
  4978.1     .05       0  4982.4      .1       0  5166.1     .07       0
Bank Sta=4978.1,4982.4
XS Rating Curve= 0 ,0
Exp/Cntr=0.3,0.1

Type RM Length L Ch R = 1 ,22799   ,426,426,426
BEGIN DESCRIPTION:
Stream0755 46.0
END DESCRIPTION:
XS GIS Cut Line= 3
      2467474.98     13661525.01        2466975.       13661875.
        2466875.     13662274.98
#Sta/Elev= 30
  4385.7  286.95  4536.1  281.91  4649.4  280.57  4769.2  280.25    4833  279.61
  4902.3  279.08  4931.9   275.7  4952.8  276.22  4959.4   275.1  4988.6  277.07
  4998.6   276.4  5006.3  272.37  5011.8  271.84  5012.1  271.34  5016.2  271.84
  5019.2  275.05  5026.9   276.3  5055.3  276.63  5119.7  275.57  5193.8  277.09
  5212.5  277.66  5225.4  276.34  5243.4  278.32  5261.4  281.67  5266.6  281.59
  5284.6  283.89  5294.9  283.93  5343.9  288.04  5360.3  288.62  5408.3  289.98
#Mann= 8 ,-1 , 0
  4385.7     .12       0  4649.4     .07       0  4769.2     .12       0
    4833      .1       0  5011.8     .05       0  5016.2      .1       0
  5193.8     .07       0  5360.3     .05       0
Bank Sta=5011.8,5016.2
XS Rating Curve= 0 ,0
Exp/Cntr=0.3,0.1

Type RM Length L Ch R = 1 ,22373   ,488,488,488
BEGIN DESCRIPTION:
Stream0755 45.0
END DESCRIPTION:
XS GIS Cut Line= 3
      2467024.97     13661225.03        2466625.       13661675.
      2466475.01     13662074.96
#Sta/Elev= 30
  4401.8  284.69  4465.7  284.48  4574.7  282.31    4699  278.67  4727.5  275.61
    4735  273.83    4763  272.66  4883.4   274.5  4978.8  274.53    4990  273.65
  4998.3   269.5  4998.6     269  5002.7   269.5  5006.5   269.5  5013.6  273.03
  5025.2  275.04  5099.1  277.44  5104.4  278.61  5129.3  277.77  5134.7  278.76
  5142.7  278.66  5184.5  276.56  5196.1  278.26  5220.1  279.71    5245  279.77
  5275.3  283.19  5300.2   282.6  5347.9  284.17  5393.4  285.97    5431  287.93
#Mann= 7 ,-1 , 0
  4401.8     .07       0  4574.7      .1       0  4978.8     .07       0
  4998.3     .05       0  5002.7     .07       0  5347.9     .05       0
  5393.4    .035       0
Bank Sta=4998.3,5002.7
XS Rating Curve= 0 ,0
Exp/Cntr=0.3,0.1

Type RM Length L Ch R = 1 ,21885   ,433,433,433
BEGIN DESCRIPTION:
Stream0755 44.0
END DESCRIPTION:
XS GIS Cut Line= 3
      2466740.32     13660905.44      2466443.16     13661339.13
        2466225.       13661875.
#Sta/Elev= 30
  4507.6  283.18    4550  282.88  4640.4  281.94  4648.1  281.74  4654.1   280.5
    4684  279.44  4731.7  278.92  4741.7  278.67  4806.5  277.19  4862.1  274.73
  4893.1  274.24  4907.1  272.72  4913.3  273.31  4935.1  271.48  4991.9  271.46
  5000.8  270.65  5013.4  267.46  5013.7  266.96  5017.9  267.46  5044.5  270.36
  5067.4  270.75  5072.8  271.58  5082.8  271.32  5091.5  269.71    5121  273.35
  5126.3  272.68  5222.6  276.28    5228  275.84  5350.4  278.57  5611.9   283.8
#Mann= 10 ,-1 , 0
  4507.6     .07       0    4550    .035       0  4731.7     .07       0
  4741.7      .1       0  4862.1    .035       0  4913.3      .1       0
  5013.4     .05       0  5017.9      .1       0  5044.5     .07       0
  5350.4     .05       0
Bank Sta=5013.4,5017.9
XS Rating Curve= 0 ,0
Exp/Cntr=0.3,0.1

Type RM Length L Ch R = 1 ,21452   ,472,472,472
BEGIN DESCRIPTION:
Stream0755 43.0
END DESCRIPTION:
XS GIS Cut Line= 3
      2466674.99       13660925.        2466325.       13660975.
      2465524.96     13661175.01
#Sta/Elev= 30
  4641.2  282.18  4698.6  280.67  4823.5  276.19  4843.2  275.59  4863.4  273.85
  4873.5  271.84  4883.6  271.27  4893.7     269  4984.6  269.95  4992.2  268.49
  4997.3  268.49  5002.8  266.61  5003.1  266.11    5007  266.11  5007.3  266.61
  5012.8  267.15  5020.1   266.7  5077.2  271.84  5108.1  271.76  5149.4  268.93
    5170   268.2  5182.9   268.5  5224.1  269.87  5293.7  274.77  5324.6  274.79
  5376.1  276.81  5383.9  276.42  5654.4  283.84  5718.9  286.11  5819.4  290.86
#Mann= 6 ,-1 , 0
  4641.2    .035       0  4698.6     .07       0  4823.5      .1       0
  5002.8     .05       0  5007.3      .1       0  5020.1     .07       0
Bank Sta=5002.8,5007.3
XS Rating Curve= 0 ,0
Exp/Cntr=0.3,0.1

Type RM Length L Ch R = 1 ,20980   ,261,261,261
BEGIN DESCRIPTION:
Stream0755 42.0
END DESCRIPTION:
XS GIS Cut Line= 3
      2466624.98       13660725.        2466025.       13660675.
      2465674.98     13660925.01
#Sta/Elev= 30
  4397.4  281.39  4398.3  281.39  4477.7  279.48  4557.9  275.84  4580.5  275.62
  4638.2  273.22  4695.9  272.38  4700.9  271.81  4794.2  271.08  4889.1  269.79
  4909.1  267.58  4949.5  268.51  4979.4  268.95  4989.4  265.57  4994.6  265.34
    4995  264.84    4999  264.84  4999.3  265.34  5002.5  265.34  5006.8     268
  5021.6  268.07  5027.7  267.32  5063.4  270.02    5099  270.79  5143.2  272.99
  5208.4  274.96  5229.3  274.97    5244   275.9  5336.2  278.36  5429.6  281.79
#Mann= 6 ,-1 , 0
  4397.4    .035       0  4398.3     .07       0  4794.2     .12       0
  4949.5     .07       0  4994.6     .05       0  4999.3     .07       0
Bank Sta=4994.6,4999.3
XS Rating Curve= 0 ,0
Exp/Cntr=0.3,0.1

Type RM Length L Ch R = 1 ,20719   ,220,220,220
BEGIN DESCRIPTION:
E21318
END DESCRIPTION:
XS GIS Cut Line= 3
      2466707.77     13660573.32      2465946.58     13660400.97
      2465185.47     13660544.58
#Sta/Elev= 30
  4344.5  280.12  4495.7  279.24    4582  277.19  4587.1     278  4624.2  275.61
  4644.7  275.68  4673.4  273.96  4678.5  274.67  4764.8  271.34    4770  271.93
  4813.1  271.12  4856.3  269.26  4899.4  268.47  4904.5  269.11  4928.7  267.94
  4952.8  266.79  4990.8   267.6  4997.6  266.45  5031.6  262.86    5032  262.36
  5036.3  262.86  5044.6  267.77  5065.1  267.24  5075.3  268.02    5173  268.28
  5335.3  270.39  5584.5  275.43  5828.7  282.76  5886.3  286.09  5899.5  286.81
#Mann= 6 ,-1 , 0
  4344.5     .07       0  4928.7     .12       0  4997.6     .07       0
  5031.6     .05       0  5036.3     .07       0  5886.3     .05       0
Bank Sta=5031.6,5036.3
XS Rating Curve= 0 ,0
Exp/Cntr=0.3,0.1

Type RM Length L Ch R = 1 ,20499   ,575,575,575
BEGIN DESCRIPTION:
Stream0755 41.0
END DESCRIPTION:
XS GIS Cut Line= 3
      2466643.93     13659765.07        2466125.       13660225.
      2464941.42     13660431.63
#Sta/Elev= 30
  4301.5  281.37  4647.8  274.58  4695.9  273.75  4803.8  270.86  4874.7  267.34
  4888.3  264.82  4902.5  267.09    4910  265.84  4941.1  266.46  5005.1   266.6
  5015.2  263.25  5024.9  262.43  5025.2  261.93  5029.6  262.43  5035.5  266.53
  5055.8  267.68  5126.9  267.69  5157.3   265.3  5248.7  267.58  5421.3  267.88
  5476.6  269.62  5528.9  270.02  5817.2  277.29  5986.3  284.24  6073.3  288.35
  6101.4  287.33  6127.8  291.21  6132.8  289.99  6152.2  292.64  6196.4  293.34
#Mann= 9 ,-1 , 0
  4301.5     .05       0  4647.8    .035       0  4695.9      .1       0
  4941.1     .07       0  5024.9     .05       0  5029.6     .07       0
  5476.6    .035       0  5528.9     .07       0  5986.3     .05       0
Bank Sta=5024.9,5029.6
XS Rating Curve= 0 ,0
Exp/Cntr=0.3,0.1

Type RM Length L Ch R = 1 ,19924   ,412,412,412
BEGIN DESCRIPTION:
Stream0755 40.0
END DESCRIPTION:
XS GIS Cut Line= 3
      2466224.98     13659625.02      2465808.72     13659989.94
      2464965.46     13660359.37
#Sta/Elev= 30
  4431.2  274.52  4587.3  271.57  4622.4  271.87  4693.6  269.25  4789.7   267.5
  4849.2  267.16  4920.4  265.01  4983.9  265.55  4997.2  258.82  4997.5  258.32
  5002.3  258.82  5007.5  263.25    5013  265.05  5039.4  264.13  5083.1  262.71
  5088.6  263.63    5098  262.09  5119.8   266.4  5141.7  266.39  5164.2  269.49
  5194.5  269.82  5447.4  270.81  5461.1   269.7  5484.5  273.27  5512.2  274.05
  5643.9   277.6  5682.4   281.1  5743.5  283.69  5862.4  290.84  5905.4  291.66
#Mann= 8 ,-1 , 0
  4431.2     .05       0  4789.7      .1       0  4997.2     .05       0
  5002.3      .1       0  5039.4     .07       0  5194.5    .035       0
  5512.2     .07       0  5743.5     .05       0
Bank Sta=4997.2,5002.3
XS Rating Curve= 0 ,0
Exp/Cntr=0.3,0.1

Type RM Length L Ch R = 1 ,19512   ,377,377,377
BEGIN DESCRIPTION:
Stream0755 39.0
END DESCRIPTION:
XS GIS Cut Line= 3
      2466124.96     13659625.01      2465736.44      13659668.7
      2465024.97     13659925.01
#Sta/Elev= 30
  4555.9  272.72  4775.9  266.91  4868.9  265.66  4928.2  265.51  4945.1   264.4
    4959  264.86  4977.6   263.1  4982.9  260.12  4990.9  257.67  4998.9  256.72
  4999.3  256.22  5004.1  256.72  5008.3  263.83  5095.1   262.1  5139.1  264.39
  5224.8  263.98  5235.4  264.72  5243.2  270.29  5248.5   265.9  5256.6  264.82
  5301.4  264.97    5330  266.55  5335.3   267.5  5373.6  267.74  5416.1  269.53
  5452.8  271.79  5490.5  275.43  5531.9  277.58    5657  285.21  5703.1  287.27
#Mann= 7 ,-1 , 0
  4555.9     .05       0  4868.9      .1       0  4998.9     .05       0
  5004.1      .1       0  5139.1     .07       0  5301.4    .035       0
  5531.9     .07       0
Bank Sta=4998.9,5004.1
XS Rating Curve= 0 ,0
Exp/Cntr=0.3,0.1

Type RM Length L Ch R = 1 ,19135   ,418,418,418
BEGIN DESCRIPTION:
Stream0755 38.0
END DESCRIPTION:
XS GIS Cut Line= 3
      2466025.03     13659374.99        2465525.       13659525.
      2465124.95     13659675.02
#Sta/Elev= 30
  4471.2  274.25    4513  273.59  4544.3  269.25  4591.8  267.31  4767.9   264.3
  4797.4  263.07  4826.2     264  4867.1  262.86  4878.4  263.24  4888.8  262.68
  4899.3  259.89  4905.4   259.8  4920.2  262.37  4971.5  261.78  4982.8  262.52
  5014.6  262.44  5025.3  261.65  5033.3     257  5034.6  257.02  5044.1  256.58
  5044.5  256.08  5049.3  256.58  5063.6  262.37  5093.8  262.44  5132.1  261.08
  5196.2  263.34  5259.4  268.75  5350.1  272.63  5388.4  276.27  5420.5  278.31
#Mann= 6 ,-1 , 0
  4471.2     .05       0  4591.8     .15       0  4797.4      .1       0
  5034.6     .07       0  5044.1     .05       0  5049.3     .07       0
Bank Sta=5044.1,5049.3
XS Rating Curve= 0 ,0
Exp/Cntr=0.3,0.1

Type RM Length L Ch R = 1 ,18717   ,424,424,424
BEGIN DESCRIPTION:
Stream0755 37.0
END DESCRIPTION:
XS GIS Cut Line= 3
      2465924.99       13659275.        2465525.       13659275.
        2465125.       13659575.
#Sta/Elev= 30
  4599.8  274.32  4609.8  273.41  4639.8  268.73  4659.8  266.47  4689.8  265.56
  4699.8  265.84  4719.8  264.88  4745.1  264.82  4843.5  263.62  4939.8  262.29
  4949.8  258.65  4957.1  253.48  4957.5  252.98    4962  252.98  4962.4  253.48
  5002.9  254.06  5013.3  258.92  5021.7  257.08  5027.9  257.29  5036.3  259.49
  5041.5  259.38  5049.8  260.81  5093.1  260.45  5127.9  261.75  5227.9  262.82
  5321.7  265.97  5327.9   265.8  5442.5  272.08  5457.1  273.46  5499.8  275.76
#Mann= 6 ,-1 , 0
  4599.8     .05       0  4745.1     .15       0  4843.5      .1       0
  4957.1     .05       0  4962.4      .1       0  5093.1     .07       0
Bank Sta=4957.1,4962.4
XS Rating Curve= 0 ,0
Exp/Cntr=0.3,0.1

Type RM Length L Ch R = 1 ,18293   ,471,471,471
BEGIN DESCRIPTION:
Stream0755 36.0
END DESCRIPTION:
XS GIS Cut Line= 3
      2465524.99     13658175.02        2465275.       13658975.
      2465025.02     13659374.98
#Sta/Elev= 30
  4161.9  275.46  4319.8  270.87    4351  268.67  4423.8  268.52  4475.7  266.98
  4480.9  265.16  4507.6  263.67  4518.6  261.11    4539  260.17  4558.8  261.44
  4611.6  260.55  4648.5   258.9  4713.9  258.37  4718.7  257.52    4746  258.24
  4751.2  259.59  4832.4  260.35  4951.3  260.13  4958.1  255.63  4965.9     253
  4966.3   252.5  4971.2     253  4983.8  255.25    5003  256.07  5007.7  260.06
  5023.1  260.69  5044.3  259.38  5138.6  260.34  5313.8  266.42  5471.7  273.73
#Mann= 9 ,-1 , 0
  4161.9     .05       0  4319.8     .07       0  4558.8     .12       0
  4611.6     .07       0  4713.9     .15       0  4965.9     .05       0
  4971.2     .15       0  5023.1     .07       0  5313.8     .05       0
Bank Sta=4965.9,4971.2
XS Rating Curve= 0 ,0
Exp/Cntr=0.3,0.1

Type RM Length L Ch R = 1 ,17822   ,448,448,448
BEGIN DESCRIPTION:
Stream0755 35.0
END DESCRIPTION:
XS GIS Cut Line= 3
      2465525.02     13658024.98        2464925.       13658825.
      2464775.01     13659174.98
#Sta/Elev= 30
  4004.4  279.84  4290.9  268.83  4397.1  262.82  4476.9  260.49  4597.5  258.99
  4647.1  259.79  4661.7  259.13  4676.3  259.46  4697.1  256.05  4704.4  252.52
  4711.7  256.02  4726.3  257.94  4805.7  259.09  4882.6  258.39  4947.1  258.77
  4979.2  257.79  4990.9  256.58  4994.5  252.45  4994.9  251.95  4999.8  252.45
  5013.5  253.93  5026.2  253.14  5037.1  256.01  5047.9  253.19  5058.8  256.61
  5066.1  259.79  5071.5  259.35  5102.3  261.19  5219.7  264.07  5385.2  268.27
#Mann= 8 ,-1 , 0
  4004.4     .05       0  4476.9     .12       0  4597.5      .1       0
  4805.7     .15       0  4979.2     .07       0  4994.5     .05       0
  4999.8     .07       0  5219.7     .05       0
Bank Sta=4994.5,4999.8
XS Rating Curve= 0 ,0
Exp/Cntr=0.3,0.1

Type RM Length L Ch R = 1 ,17374   ,457,457,457
BEGIN DESCRIPTION:
Stream0755 34.0
END DESCRIPTION:
XS GIS Cut Line= 3
      2465624.97     13657675.03        2464825.       13658475.
      2464274.97     13659075.03
#Sta/Elev= 30
  3868.2   293.4  4045.2  286.82  4094.4  284.69  4221.7  277.56  4270.3   275.6
    4448  267.83    4646  261.55  4722.6  259.91  4865.8  257.32  4928.8   258.1
  4971.2  257.91  4985.4  257.15  4992.8  252.61  4993.3  252.11  4998.6  252.11
  4999.1  252.61  5013.4  254.11  5020.8  257.27    5035  257.71  5055.9  257.02
  5096.8  256.97  5204.5  257.69  5254.5  259.19  5275.5  258.76  5370.1  259.43
  5417.3  259.56  5501.8  261.99  5686.1  265.62  5728.7   267.2  5813.5  268.26
#Mann= 9 ,-1 , 0
  3868.2     .05       0  4045.2     .07       0  4270.3     .05       0
  4722.6     .12       0  4865.8      .1       0  4992.8     .05       0
  4999.1      .1       0  5096.8     .07       0  5370.1     .05       0
Bank Sta=4992.8,4999.1
XS Rating Curve= 0 ,0
Exp/Cntr=0.3,0.1

Type RM Length L Ch R = 1 ,16917   ,451,451,451
BEGIN DESCRIPTION:
Stream0755 33.0
END DESCRIPTION:
XS GIS Cut Line= 3
      2464925.01     13657774.99        2464725.       13658125.
        2464225.     13659025.01
#Sta/Elev= 30
  4589.8  278.65  4780.6  266.05  4878.5  261.11  4904.4  259.28  4935.3  258.25
  4947.6  256.94  4957.7  257.38  4963.4  254.99  4979.3  253.33    4985  256.11
  4995.8  255.86  5000.9  254.73  5006.7  256.06  5015.8  253.33  5028.4  254.19
  5035.5  253.12    5036  252.62  5041.9  253.12  5050.1  255.58  5087.9  256.48
  5131.3  254.96  5206.8  256.83  5328.6   256.4  5404.8  255.52  5465.5  256.99
  5610.7  258.62  5721.6   261.9  5759.4  262.09  5905.8  266.53  6022.5  268.19
#Mann= 6 ,-1 , 0
  4589.8     .05       0  4878.5      .1       0  5035.5     .05       0
  5041.9      .1       0  5328.6     .07       0  5465.5     .05       0
Bank Sta=5035.5,5041.9
XS Rating Curve= 0 ,0
Exp/Cntr=0.3,0.1

Type RM Length L Ch R = 1 ,16466   ,462,462,462
BEGIN DESCRIPTION:
Stream0755 32.0
END DESCRIPTION:
XS GIS Cut Line= 3
      2464824.98     13657425.03        2464325.       13658225.
      2464124.99     13658925.03
#Sta/Elev= 30
  4064.9  295.39  4083.2  294.58  4203.4     287  4370.9  277.59  4507.7  268.17
  4613.6  262.21  4725.2  256.46  4775.4  255.39  4842.6  255.35  4848.5  254.23
  4861.1  254.08  4913.9  254.24  4942.8  252.46  4991.4  252.46  4997.3  252.43
  4997.8  251.93  5003.3  251.93  5003.8  252.43  5025.2  253.01  5030.4   252.6
  5039.5  254.96  5063.3  254.91  5153.9  254.21  5232.8  254.97  5372.3  257.42
  5382.7  258.24    5423  258.86  5621.9  265.48  5694.7  267.19  5736.3  267.46
#Mann= 9 ,-1 , 0
  4064.9     .07       0  4083.2     .05       0  4613.6     .07       0
  4861.1      .1       0  4991.4     .05       0  4997.3     .05       0
  5003.8     .05       0  5063.3     .07       0  5232.8     .05       0
Bank Sta=4997.3,5003.8
XS Rating Curve= 0 ,0
Exp/Cntr=0.3,0.1

Type RM Length L Ch R = 1 ,16004   ,433,433,433
BEGIN DESCRIPTION:
Stream0755 31.0
END DESCRIPTION:
XS GIS Cut Line= 3
      2464074.98     13657775.04        2463925.       13658075.
        2463975.     13658725.01
#Sta/Elev= 30
  4664.2  261.74  4678.2  261.57  4694.9  261.28  4731.2  253.06  4798.3  251.39
  4851.4  252.75  4879.4  252.95  4896.2  252.45  4910.4   253.1  4968.8   253.8
  4977.2  253.34  4985.6  248.98  4991.2  251.09  4993.5  246.29    4994  245.79
  4999.5  245.79    5000  246.29  5009.6  246.38  5019.6  253.49  5029.7  254.25
  5069.8  254.31  5127.4  252.86    5150  252.37    5160  252.91  5170.1  252.61
  5260.3  254.12  5270.4  254.69  5330.5  255.06  5390.7  256.37  5651.5  264.37
#Mann= 6 ,-1 , 0
  4664.2    .035       0  4678.2     .15       0  4910.4      .1       0
  4993.5     .05       0    5000      .1       0  5127.4     .05       0
Bank Sta=4993.5,5000
XS Rating Curve= 0 ,0
Exp/Cntr=0.3,0.1

Type RM Length L Ch R = 1 ,15571   ,472,472,472
BEGIN DESCRIPTION:
Stream0755 30.0
END DESCRIPTION:
XS GIS Cut Line= 3
        2464025.       13657725.        2463625.       13657875.
        2463375.       13658475.
#Sta/Elev= 30
  4566.4  261.26  4636.7  259.84    4667  252.64    4674  251.67  4747.1  251.27
  4876.1  252.37  4983.8  252.41  4990.9  251.01  4996.3  251.01  4999.5  245.93
    5000  245.43  5006.1  245.93  5008.2  245.97  5010.9  247.27  5015.3   249.4
  5026.1  251.68  5032.1   252.2  5055.9  252.56  5091.1  251.46  5114.4  252.54
  5129.5   251.4  5145.3  250.88  5177.8  251.11  5185.9  251.96  5209.7  252.48
  5244.4  251.58  5262.8  252.44  5321.3  252.61  5552.1  259.73  5643.6  261.75
#Mann= 6 ,-1 , 0
  4566.4     .05       0    4674     .15       0  4999.5     .05       0
  5006.1     .15       0  5010.9      .1       0  5129.5     .07       0
Bank Sta=4999.5,5006.1
XS Rating Curve= 0 ,0
Exp/Cntr=0.3,0.1

Type RM Length L Ch R = 1 ,15099   ,465,465,465
BEGIN DESCRIPTION:
Stream0755 29.0
END DESCRIPTION:
XS GIS Cut Line= 3
      2463632.33     13656753.51        2463225.       13657775.
      2463046.08     13658407.88
#Sta/Elev= 30
  3899.9  275.26  4038.6  271.01  4127.6  265.26  4146.5  266.01    4364  255.74
  4464.9  251.84  4649.2  248.64    4691  248.65  4720.6  244.74  4739.5  248.57
  4838.1  246.46  4847.3  247.78  4852.7  246.24  4859.7  249.15  4955.1   250.9
  4990.2  249.86  5006.7  244.33  5007.2  243.83  5013.4  244.33  5016.6  249.91
  5021.8  248.46  5041.2  250.78  5134.7   249.9  5155.5  248.13  5162.9  244.98
  5176.3  249.22  5187.9  249.14  5228.2  248.63  5572.9  259.14  5657.3  259.31
#Mann= 7 ,-1 , 0
  3899.9     .05       0    4364     .07       0  4464.9     .05       0
  4649.2      .1       0  5006.7     .05       0  5013.4      .1       0
  5187.9     .07       0
Bank Sta=5006.7,5013.4
XS Rating Curve= 0 ,0
Exp/Cntr=0.3,0.1

Type RM Length L Ch R = 1 ,14634   ,769,769,769
BEGIN DESCRIPTION:
Stream0755 28.0
END DESCRIPTION:
XS GIS Cut Line= 3
      2463475.02     13657124.98        2463075.       13657525.
        2463025.     13658325.03
#Sta/Elev= 30
  4438.5  258.44  4511.9  254.54  4552.5  253.07  4636.5  250.12  4779.2  247.74
  4947.6  248.49  4961.8  247.31  4968.9  245.09  4972.5  241.53    4973  241.03
  4979.3  241.53  5000.7  246.93  5064.3  249.15  5104.4  249.35  5114.4  248.35
  5124.4  242.65  5174.5  243.34  5184.6  248.05  5204.6  250.16  5334.9  247.07
  5344.9  242.69  5354.9  246.18  5371.2  247.25    5395  245.03  5402.5  245.37
  5407.5  248.43  5535.2  250.67  5655.5  255.08  5665.5  254.51  5805.8   257.9
#Mann= 7 ,-1 , 0
  4438.5     .05       0  4511.9     .07       0  4552.5     .05       0
  4779.2      .1       0  4972.5     .05       0  4979.3      .1       0
  5371.2     .07       0
Bank Sta=4972.5,4979.3
XS Rating Curve= 0 ,0
Exp/Cntr=0.3,0.1

Type RM Length L Ch R = 1 ,13865   ,616,616,616
BEGIN DESCRIPTION:
XS7654
END DESCRIPTION:
XS GIS Cut Line= 4
      2463118.36     13656761.53      2462708.79     13657347.77
      2462797.13     13657789.47      2462572.62     13658631.36
#Sta/Elev= 30
  4001.7  264.02  4258.4  251.11  4434.8  244.07  4481.7  245.49  4808.8  246.89
  4981.1  245.46  4996.2     238  4996.7   237.5    5003     238  5009.8  242.84
    5027  246.16  5032.1  243.71  5060.7  245.92  5083.1  245.33  5101.5  243.05
  5111.7  239.96  5118.9  242.89    5129  245.43  5142.3  246.17    5220  247.08
  5346.2  249.38  5387.1  249.44  5427.2   244.3    5445  245.79  5452.4  245.17
  5483.5  249.86  5510.3  250.53  5653.4  255.98  5829.9  260.55  6038.6  265.93
#Mann= 12 ,-1 , 0
  4001.7     .07       0  4434.8     .05       0  4808.8      .1       0
  4996.2     .05       0    5003      .1       0  5118.9     .12       0
    5220     .07       0  5346.2     .12       0    5445     .05       0
  5510.3     .07       0  5653.4     .05       0  5829.9     .07       0
Bank Sta=4996.2,5003
XS Rating Curve= 0 ,0
Exp/Cntr=0.3,0.1

Type RM Length L Ch R = 1 ,13249   ,459,459,459
BEGIN DESCRIPTION:
Stream0755 27.0
END DESCRIPTION:
XS GIS Cut Line= 3
        2463025.       13656725.        2462325.       13657525.
        2462225.     13658324.96
#Sta/Elev= 30
  3936.7  265.39  4181.9  252.49  4185.4  252.28    4369  243.78  4415.6  244.91
  4833.5  243.89  4879.7  243.38  4971.7  244.64  4992.6  243.24  4996.4  240.33
  5002.2  240.33  5006.3  235.95  5006.8  235.45  5013.3  235.95  5019.9  236.42
  5029.9  241.59  5037.5  243.31  5050.1  244.25  5105.5  244.66  5204.4  244.13
  5351.5  245.01  5382.7  245.66  5412.9  249.89  5433.1  250.87  5606.9  253.07
  5624.5  254.17  5654.8  257.87  5674.9  257.87  5695.1  259.53  5805.9  263.13
#Mann= 10 ,-1 , 0
  3936.7     .07       0  4181.9     .12       0  4185.4     .07       0
  4415.6     .05       0  4833.5      .1       0  5006.3     .05       0
  5013.3      .1       0  5105.5      .1       0  5204.4     .05       0
  5351.5     .07       0
Bank Sta=5006.3,5013.3
XS Rating Curve= 0 ,0
Exp/Cntr=0.3,0.1

Type RM Length L Ch R = 1 ,12790   ,449,449,449
BEGIN DESCRIPTION:
Stream0755 26.0
END DESCRIPTION:
XS GIS Cut Line= 3
      2462824.96     13656525.04        2462025.       13657325.
        2461375.       13658125.
#Sta/Elev= 30
  3867.7  267.32  3992.3  263.05  4323.6  249.58  4459.1  244.56  4466.2  244.16
  4560.6   241.8  4594.5  242.74  4738.9  242.29  4942.5  242.46  4956.6  241.39
  4967.2  235.61  4967.7  235.11  4974.2  235.61  4984.9   236.7  4995.5  242.25
  5000.6  242.25  5124.7  241.69    5198  238.96    5305  242.23  5397.7  242.62
  5418.5  240.21  5431.7  241.64  5439.3  238.88  5447.3  241.49  5457.8   241.5
  5482.4  242.52  5503.3  238.43  5553.1  244.86  5837.3  256.17  6029.8  261.72
#Mann= 13 ,-1 , 0
  3867.7     .07       0  3992.3     .12       0  4323.6     .07       0
  4459.1     .12       0  4466.2     .07       0  4594.5     .05       0
  4738.9      .1       0  4967.2     .05       0  4974.2      .1       0
  5000.6     .12       0  5124.7     .07       0  5431.7     .12       0
  5457.8     .07       0
Bank Sta=4967.2,4974.2
XS Rating Curve= 0 ,0
Exp/Cntr=0.3,0.1

Type RM Length L Ch R = 1 ,12341   ,436,436,436
BEGIN DESCRIPTION:
Stream0755 25.0
END DESCRIPTION:
XS GIS Cut Line= 3
      2462424.97     13656375.03        2461825.       13657075.
        2461375.     13657875.01
#Sta/Elev= 30
  4068.5  262.75  4079.4  262.52  4166.5  259.64  4235.8   257.1  4450.4  248.38
  4515.4  246.42    4673  241.09    4705  240.89  4799.6  240.98  4976.7  241.14
  4983.3  240.54  4987.1  236.67  5000.6  234.64  5001.1  234.14  5007.6  234.64
  5020.1  240.16    5101  240.82    5182  237.93  5187.7  235.53  5196.9  235.21
  5203.6  235.56  5217.9  239.68  5262.9  239.32  5277.2  236.27  5284.6  239.19
  5300.2  240.09  5380.5   240.8  5468.2  243.86  5667.3  246.62  5908.3  255.02
#Mann= 13 ,-1 , 0
  4068.5     .12       0  4079.4     .07       0  4166.5     .12       0
  4235.8     .07       0  4450.4     .12       0  4515.4     .07       0
    4673     .05       0    4705     .07       0  4799.6      .1       0
  5000.6     .05       0  5007.6      .1       0  5217.9     .12       0
  5380.5     .07       0
Bank Sta=5000.6,5007.6
XS Rating Curve= 0 ,0
Exp/Cntr=0.3,0.1

Type RM Length L Ch R = 1 ,11905   ,426,426,426
BEGIN DESCRIPTION:
Stream0755 24.0
END DESCRIPTION:
XS GIS Cut Line= 3
      2462274.99     13656225.01        2461475.       13657025.
      2461174.97     13657425.03
#Sta/Elev= 30
  3864.1  262.27  4016.2  255.09  4186.5  247.32  4365.8  241.13  4440.1  239.75
  4458.1   239.2    4509  239.84    4656   239.3  4684.3   237.8  4712.6  238.81
  4795.5  237.67  4825.8  237.08  4868.2  238.47  4981.3  238.79  4998.6  238.12
  5002.7  236.08  5005.2  233.66  5005.7  233.16  5012.8  233.66  5031.9  239.01
    5059  239.39  5098.5  238.04  5103.9  237.36  5123.6   236.7  5145.5   238.6
  5152.7  239.99    5159  239.27  5167.3  240.33  5223.6  242.56  5495.5  249.43
#Mann= 11 ,-1 , 0
  3864.1     .12       0  4016.2     .07       0  4186.5     .12       0
  4365.8     .05       0  4440.1     .07       0    4509     .05       0
  4795.5      .1       0  5005.2     .05       0  5012.8      .1       0
  5098.5     .12       0  5103.9     .07       0
Bank Sta=5005.2,5012.8
XS Rating Curve= 0 ,0
Exp/Cntr=0.3,0.1

Type RM Length L Ch R = 1 ,11479   ,449,449,449
BEGIN DESCRIPTION:
Stream0755 23.0
END DESCRIPTION:
XS GIS Cut Line= 3
      2462024.99     13656125.01        2461225.       13656775.
      2460975.02     13656874.99
#Sta/Elev= 30
  3974.2  251.91  4051.7  246.64    4130  243.55    4138  242.35  4187.5  240.13
  4280.2  238.57  4556.7  237.67  4643.3  236.23    4699  234.72  4721.3  236.29
  4762.9  237.06  4849.1  236.71  4869.9  235.72  4890.7  237.48  4948.2   237.9
  4962.6  236.15    4969  231.79    4977  230.71  4983.4  231.69  4987.5  230.28
    4988  229.78  4995.2  230.28  5001.7  236.65  5037.3  236.65  5097.9   240.1
  5127.5  240.29  5134.2  241.13  5181.3  242.18  5189.3  243.17  5274.2  246.37
#Mann= 5 ,-1 , 0
  3974.2     .05       0  4643.3      .1       0  4987.5     .05       0
  4995.2      .1       0  5189.3    .035       0
Bank Sta=4987.5,4995.2
XS Rating Curve= 0 ,0
Exp/Cntr=0.3,0.1

Type RM Length L Ch R = 1 ,11030   ,433,433,433
BEGIN DESCRIPTION:
Stream0755 22.0
END DESCRIPTION:
XS GIS Cut Line= 3
      2461975.03     13656074.99        2461175.       13656375.
      2460580.56     13656488.47
#Sta/Elev= 30
  4145.2   249.7  4356.2  238.67    4720  235.25  4775.4  234.91  4807.4  232.92
  4826.2  234.62  4914.2  236.37  4946.2  235.09  4967.6  235.95  4978.3   232.8
  4984.5  227.86  4993.1  227.42  4993.6  226.92  5000.9  227.42  5002.2  227.42
  5009.8  233.07    5020  234.48  5030.8  232.37  5040.4  235.28  5077.8  236.72
  5129.9     237    5135  235.25  5152.3   234.8    5182   236.4  5187.1  235.68
  5213.4  242.69  5229.8  244.27  5291.4   246.4  5584.1  248.68  5604.8  248.91
#Mann= 7 ,-1 , 0
  4145.2     .05       0    4720     .15       0  4826.2      .1       0
  4993.1     .05       0  5000.9      .1       0  5229.8    .035       0
  5584.1     .05       0
Bank Sta=4993.1,5000.9
XS Rating Curve= 0 ,0
Exp/Cntr=0.3,0.1

Type RM Length L Ch R = 1 ,10597   ,466,466,466
BEGIN DESCRIPTION:
Stream0755 21.0
END DESCRIPTION:
XS GIS Cut Line= 3
      2462024.98       13656025.        2461225.       13656025.
      2460669.43     13656149.86
#Sta/Elev= 30
  4204.8  252.07  4284.8  248.52  4444.8  239.78  4504.8  237.75  4584.8  236.17
  4785.7  234.69  4814.8  234.02  4874.8   234.2  4884.1  233.26  4904.8  230.67
  4914.8  230.51  4924.8  232.18  4954.8  234.13  4994.8  233.77  5002.3  226.23
  5011.1  225.71  5011.6  225.21  5018.9  225.71  5023.9   231.4    5029  230.91
  5035.5  234.22  5045.8   234.1    5056  235.03  5126.9  235.24  5189.3  235.32
  5230.3  236.21  5279.1  238.42  5445.5   244.8  5487.6  245.57  5574.2  244.89
#Mann= 7 ,-1 , 0
  4204.8     .05       0  4785.7     .15       0  4884.1      .1       0
  5011.1     .05       0  5018.9      .1       0  5126.9     .07       0
  5279.1    .035       0
Bank Sta=5011.1,5018.9
XS Rating Curve= 0 ,0
Exp/Cntr=0.3,0.1

Type RM Length L Ch R = 1 ,10131   ,485,485,485
BEGIN DESCRIPTION:
Stream0755 20.0
END DESCRIPTION:
XS GIS Cut Line= 3
      2461725.02     13655374.99        2461325.       13655625.
      2460675.04     13655874.99
#Sta/Elev= 30
  4522.1  240.47  4624.1  236.01  4837.2  231.33  4864.1  231.03  4928.4   233.7
  4943.7  231.26  4949.6  233.73  4955.4  233.24  4958.4  232.99  4970.8  229.08
  4986.2  232.54  4996.5  231.93  5003.5  226.95  5008.8  229.26  5011.3  224.38
  5011.8  223.88  5019.3  224.38    5026  226.61  5033.5  232.44  5038.8  231.02
  5047.4  234.07  5063.7  233.97  5172.3  233.46    5267  233.17  5278.9  233.32
    5312  231.94  5317.4  232.89  5385.5  233.64  5590.6  242.11  5690.2  245.39
#Mann= 10 ,-1 , 0
  4522.1     .05       0  4837.2     .15       0  4955.4      .1       0
  5011.3     .05       0  5019.3      .1       0  5063.7    .035       0
  5172.3     .12       0    5267      .1       0  5278.9     .12       0
  5385.5    .035       0
Bank Sta=5011.3,5019.3
XS Rating Curve= 0 ,0
Exp/Cntr=0.3,0.1

Type RM Length L Ch R = 1 ,9646    ,670,670,670
BEGIN DESCRIPTION:
Stream0755 19.0
END DESCRIPTION:
XS GIS Cut Line= 3
      2461990.01     13655015.46        2461325.       13655175.
      2460575.02     13655724.98
#Sta/Elev= 30
  4316.2  250.77  4352.2  252.04  4425.4  250.21  4551.4   244.9  4677.4  237.83
  4803.4  232.52  4829.3  232.17  4866.4  229.88  4892.5  229.79  4917.8  231.46
  4958.9  231.53  4969.2  226.73  4972.5  222.04    4973  221.54  4980.5  222.04
  4989.8  222.96  4997.5  229.76  5003.2  229.76  5007.4  231.25  5099.3  230.57
  5113.9  231.85    5146  231.67  5340.9  231.97  5429.6  232.38  5444.2   231.2
  5471.3  232.18  5515.3  231.63  5590.5  233.52    5858   243.8  5930.1  245.09
#Mann= 7 ,-1 , 0
  4316.2     .07       0  4829.3      .1       0  4972.5     .05       0
  4980.5      .1       0    5146    .035       0  5340.9     .12       0
  5590.5    .035       0
Bank Sta=4972.5,4980.5
XS Rating Curve= 0 ,0
Exp/Cntr=0.3,0.1

Type RM Length L Ch R = 1 ,8976    ,700,700,700
BEGIN DESCRIPTION:
E21317
END DESCRIPTION:
XS GIS Cut Line= 4
      2461968.48     13654764.13      2461595.08     13654749.77
      2461099.62     13654900.57      2460489.67     13655288.06
#Sta/Elev= 30
  4706.9  245.88    4810  245.39  4860.5  243.78  4940.5  240.38  4950.6  236.76
  4960.6  236.62  4970.6  239.02  4980.6   231.2  4986.5  221.54    4987  221.04
  4994.6  221.54  4998.6  221.59  5020.6  227.28  5050.6  228.86  5122.5  227.78
  5187.4  228.95    5215  228.21    5227  229.36    5342  228.37  5389.7   229.5
  5436.1  228.48  5512.8  229.83  5619.2  229.59  5728.1  230.02  5779.8  231.41
  5785.7  230.64  5896.1  230.78  5964.6  232.08  6031.4  232.83  6321.1  241.68
#Mann= 8 ,-1 , 0
  4706.9     .07       0  4986.5     .05       0  4994.6     .07       0
  4998.6      .1       0  5512.8     .12       0  5619.2     .07       0
  5896.1     .12       0  5964.6    .035       0
Bank Sta=4986.5,4994.6
XS Rating Curve= 0 ,0
Exp/Cntr=0.3,0.1

Type RM Length L Ch R = 1 ,8276    ,473,473,473
BEGIN DESCRIPTION:
Stream0755 18.0
END DESCRIPTION:
XS GIS Cut Line= 3
      2461724.97     13654175.02        2461175.       13654525.
      2460475.03     13655124.98
#Sta/Elev= 30
  4348.4  237.66  4580.3   228.4  4659.1  227.55  4718.7  228.17    4941  228.56
  4964.7  225.85  4971.5   219.5  4973.4  218.82  4973.9  218.32  4981.5  218.82
  4986.7  219.49  4992.7   224.2  4997.3  225.95  5056.8   226.2  5092.5  228.54
  5110.7   227.5    5149  226.97  5175.1  228.68  5369.1  229.46  5376.2  230.23
  5404.7  229.28  5553.5   229.8  5642.1  231.36  5709.9  233.31  5724.1  234.77
    5761  235.36    5775  235.88  5907.5  240.01  5907.9  240.02  5922.2  240.15
#Mann= 11 ,-1 , 0
  4348.4     .07       0  4718.7      .1       0  4973.4     .05       0
  4981.5      .1       0  5110.7     .12       0  5175.1     .07       0
  5642.1    .035       0    5761     .07       0    5775     .05       0
  5907.5    .035       0  5907.9     .05       0
Bank Sta=4973.4,4981.5
XS Rating Curve= 0 ,0
Exp/Cntr=0.3,0.1

Type RM Length L Ch R = 1 ,7803    ,464,464,464
BEGIN DESCRIPTION:
Stream0755 17.0
END DESCRIPTION:
XS GIS Cut Line= 3
        2461675.       13654125.        2461075.       13654225.
      2460524.98     13654525.01
#Sta/Elev= 30
  4392.6  236.61  4547.2  231.21  4656.2  226.07  4676.5  227.02  4724.6  227.38
  4848.2   226.7  4919.8  227.29    4973  226.57  4980.6  225.82  4990.7  221.88
  4994.3  217.56  4994.8  217.06  5002.4  217.56  5014.6  217.57  5023.7  220.93
  5030.8   224.9  5036.5   223.3  5046.4  225.78  5083.8     226  5103.4  227.26
  5197.7  227.31  5331.2  227.07    5363     226  5390.5   227.4  5412.4  227.13
  5468.9  228.32  5488.3  229.66  5502.1  229.23  5603.3  232.99  5627.4  233.47
#Mann= 8 ,-1 , 0
  4392.6     .07       0  4848.2      .1       0  4994.3     .05       0
  5002.4      .1       0  5083.8     .12       0  5197.7     .07       0
  5468.9     .12       0  5603.3     .07       0
Bank Sta=4994.3,5002.4
XS Rating Curve= 0 ,0
Exp/Cntr=0.3,0.1

Type RM Length L Ch R = 1 ,7339    ,423,423,423
BEGIN DESCRIPTION:
Stream0755 16.0
END DESCRIPTION:
XS GIS Cut Line= 3
      2461625.02       13654025.        2460975.       13653925.
        2460175.       13653825.
#Sta/Elev= 30
  4342.6  235.22  4605.7  226.17  4757.2  226.22    4889  225.93  4939.6   222.9
    4980  224.04  4993.7  216.83  4994.2  216.33  5001.8  216.83  5010.3  222.48
  5020.4  224.05    5062  225.64  5160.9  224.63  5191.7  222.89  5263.1  222.93
  5322.8  224.89  5360.6  224.12  5373.1  225.97  5457.3  225.87  5473.9   226.1
    5484  220.74  5494.1  224.73  5514.2  222.77  5521.8  224.03  5526.8  221.95
  5534.4  224.83  5544.5  225.95  5655.3  226.94  5751.1  230.74  5806.5   233.5
#Mann= 9 ,-1 , 0
  4342.6     .07       0  4757.2      .1       0  4993.7     .05       0
  5001.8      .1       0    5062     .12       0  5160.9     .07       0
  5263.1    .035       0  5457.3     .12       0  5751.1     .05       0
Bank Sta=4993.7,5001.8
XS Rating Curve= 0 ,0
Exp/Cntr=0.3,0.1

Type RM Length L Ch R = 1 ,6916    ,455,455,455
BEGIN DESCRIPTION:
Stream0755 15.0
END DESCRIPTION:
XS GIS Cut Line= 3
      2461575.03     13653925.02        2460975.       13653575.
      2460174.96     13653274.99
#Sta/Elev= 30
  4305.3  233.52  4572.1  225.84  4722.5  225.31    4780  225.75  4794.5  224.07
    4816  225.72  4839.5  225.03  4874.7  224.33  4896.2  222.36  4911.9  224.14
  5015.1  223.03  5021.3  217.15  5027.9  216.53  5028.4  216.03  5036.1  216.53
    5040  223.31  5070.3  223.91  5224.2  221.96  5271.4  223.22  5288.3   218.4
  5296.3  220.35  5301.7  218.26  5320.4  221.98  5366.4  222.83  5370.2  222.86
  5522.4  223.16  5588.3  224.54  5638.1  227.54  5747.6  230.75  5854.4  238.21
#Mann= 8 ,-1 , 0
  4305.3     .07       0  4572.1     .12       0  4722.5    .035       0
  4839.5      .1       0  5027.9     .05       0  5036.1      .1       0
  5366.4     .07       0  5370.2     .05       0
Bank Sta=5027.9,5036.1
XS Rating Curve= 0 ,0
Exp/Cntr=0.3,0.1

Type RM Length L Ch R = 1 ,6461    ,443,443,443
BEGIN DESCRIPTION:
Stream0755 14.0
END DESCRIPTION:
XS GIS Cut Line= 4
      2461584.49     13653878.46      2461118.67     13653292.16
        2460825.       13653175.      2460024.96       13653225.
#Sta/Elev= 30
  3940.7  233.06  4214.1  227.52  4342.8  225.27  4583.7  224.54  4697.1  223.15
  4721.4  220.88  4745.6  220.84  4758.1  223.18  4790.4  220.56  4835.8  222.67
    4898  223.21  4907.3  220.57  4912.7  223.15    4937  215.54  4942.4  220.51
  4961.2  217.62  4966.6  221.03  4979.6  215.18  4980.1  214.68  4988.7  215.18
  4990.9  217.67  4996.3  215.28    5003  220.85  5015.7  222.82  5045.8  220.74
  5132.1  222.01  5243.7  220.29  5416.5   224.7  5788.5  245.99  5807.3   247.6
#Mann= 8 ,-1 , 0
  3940.7     .07       0  4214.1    .035       0  4342.8     .12       0
  4835.8      .1       0  4979.6     .05       0  4988.7      .1       0
  5132.1     .05       0  5788.5     .07       0
Bank Sta=4979.6,4988.7
XS Rating Curve= 0 ,0
Exp/Cntr=0.3,0.1

Type RM Length L Ch R = 1 ,6018    ,448,448,448
BEGIN DESCRIPTION:
Stream0755 13.0
END DESCRIPTION:
XS GIS Cut Line= 3
      2461374.99     13652025.02        2460825.       13652775.
      2460024.96     13653175.02
#Sta/Elev= 30
  4064.7  230.13  4107.5  230.66  4122.2  228.82    4187  228.73  4201.1  226.57
    4260  226.42  4260.9  226.39  4527.5  220.66  4579.9  221.08  4594.5  219.85
  4738.6  221.03  4822.2  221.33  4866.2  220.11  4972.7  221.94  4987.4  220.08
  4991.6  215.12  4997.2  214.03  4997.7  213.53  5009.1  214.03  5017.1  219.09
  5031.1  221.41  5120.5  220.14    5180  220.93  5189.6     221  5350.7  220.02
  5383.2  222.47  5433.6  222.56  5562.1  227.78  5651.6  234.18  5889.2  246.98
#Mann= 10 ,-1 , 0
  4064.7     .07       0    4260    .035       0  4260.9     .12       0
  4527.5     .07       0  4738.6      .1       0  4997.2     .05       0
  5009.1      .1       0    5180     .05       0  5189.6      .1       0
  5350.7     .05       0
Bank Sta=4997.2,5009.1
XS Rating Curve= 0 ,0
Exp/Cntr=0.3,0.1

Type RM Length L Ch R = 1 ,5570    ,479,479,479
BEGIN DESCRIPTION:
Stream0755 12.0
END DESCRIPTION:
XS GIS Cut Line= 3
      2461275.04     13651924.97        2460475.       13652575.
        2460125.       13652875.
#Sta/Elev= 30
  3968.7   230.3  4118.2  227.27  4182.1  223.48    4213  223.54  4252.5  221.73
  4363.9  219.76  4514.8  219.45    4630  218.09  4679.1  219.67  4728.9  218.78
  4736.6   217.5  4759.8  219.15  4885.3  219.16  4942.8  220.57  4957.2  218.98
  4963.6   219.5  4971.5  216.86    4978  216.66  4986.4  213.16  4986.9  212.66
  4998.3  213.16  5002.8  214.24  5006.7  220.09  5070.3  220.19  5113.1  218.16
  5124.2  218.89  5141.7  219.25  5155.9   221.2    5269  224.75  5460.5   235.7
#Mann= 9 ,-1 , 0
  3968.7     .07       0    4213    .035       0  4363.9     .12       0
  4514.8     .07       0    4630     .12       0  4759.8      .1       0
  4986.4     .05       0  4998.3      .1       0  5124.2     .05       0
Bank Sta=4986.4,4998.3
XS Rating Curve= 0 ,0
Exp/Cntr=0.3,0.1

Type RM Length L Ch R = 1 ,5091    ,445,445,445
BEGIN DESCRIPTION:
Stream0755 11.0
END DESCRIPTION:
XS GIS Cut Line= 3
      2461075.01     13651674.99        2460275.       13652175.
      2459875.02       13652275.
#Sta/Elev= 30
  4056.1  229.18  4106.2   228.1  4310.2  219.55  4336.1  219.47  4346.8  218.34
  4441.1  217.02  4527.4  218.03  4563.2  218.93  4577.9  217.84  4635.7  218.21
  4666.4   217.1  4708.8  218.04  4751.9  216.48  4766.6  217.79  4818.5  217.11
  4949.4  219.25  4964.1  218.86  4970.6   214.1  4976.5  214.92  4979.9  211.98
  4980.4  211.48  4991.9  211.98  4996.6  213.94  5002.1  213.94  5009.8   219.2
  5102.1  219.46  5223.4   224.3  5270.1  225.58  5400.5  232.88  5411.8  233.36
#Mann= 8 ,-1 , 0
  4056.1     .07       0  4336.1     .12       0  4527.4      .1       0
  4979.9     .05       0  4991.9      .1       0  5102.1     .05       0
  5223.4     .07       0  5400.5     .05       0
Bank Sta=4979.9,4991.9
XS Rating Curve= 0 ,0
Exp/Cntr=0.3,0.1

Type RM Length L Ch R = 1 ,4646    ,475,475,475
BEGIN DESCRIPTION:
Stream0755 10.0
END DESCRIPTION:
XS GIS Cut Line= 3
        2461075.       13651625.        2460175.       13651825.
      2459775.04     13652074.97
#Sta/Elev= 30
  4087.5  229.46  4179.7  227.49  4230.9  224.25  4383.3  218.19  4437.1  216.76
  4490.7  216.61  4599.7  217.17  4609.9  215.29  4621.5  215.08  4630.4  215.16
  4640.7  216.65  4671.4  217.36  4693.6   216.9  4805.9   218.7  4844.3  218.07
    4948  218.59  4979.1  210.97  4979.6  210.47  4991.1  210.97  4999.2  212.83
  5017.1  211.69    5023  217.18  5038.3  218.13  5103.8  216.05    5148  218.74
  5232.4  221.57  5243.2  221.84  5412.6   230.7    5431  232.46  5481.1  234.76
#Mann= 8 ,-1 , 0
  4087.5     .07       0  4490.7     .12       0  4693.6      .1       0
  4979.1     .05       0  4991.1      .1       0  5232.4     .05       0
  5243.2     .07       0  5412.6     .05       0
Bank Sta=4979.1,4991.1
XS Rating Curve= 0 ,0
Exp/Cntr=0.3,0.1
