--- Stream0804.prj (project) ---

Proj Title=Stream0804 Base Level Engineering
Current Plan=p01
Default Exp/Contr=0.3,0.1
English Units
Geom File=g01
Flow File=f01
Plan File=p01
Y Axis Title=Elevation
X Axis Title(PF)=Main Channel Distance
X Axis Title(XS)=Station
BEGIN DESCRIPTION:
Stream0804
END DESCRIPTION:
DSS Export Rating Curves= 0
DSS Export Rating Curve Sorted= 0
DSS Export Volume Flow Curves= 0
DXF OffsetX= 0
DXF OffsetY= 0
DXF ScaleX= 1
DXF ScaleY= 10

--- Stream0804.p01 (plan) ---

Plan Title=Multiple Run
Short Identifier=Multiple
Geom File=g01
Flow File=f01
Subcritical Flow
K Sum by GR= 0
Std Step Tol= 0.01
Critical Tol= 0.01
Num of Std Step Trials= 20
Max Error Tol= 0.3
Flow Tol Ratio= 0.001
Split Flow NTrial= 30
Split Flow Tol= 0.02
Split Flow Ratio= 0.02
Log Output Level= 0
Friction Slope Method= 1
Unsteady Friction Slope Method= 2
Unsteady Bridges Friction Slope Method= 1
Parabolic Critical Depth
Global Vel Dist=  1 , 1 , 1
Global Log Level= 0
CheckData=True
Encroach Param= -1, 0, 0, 0
BEGIN DESCRIPTION:
Multiple Run
END DESCRIPTION:

--- Stream0804.f01 (steady flow) ---

Flow Title=Multiple
Number of Profiles=7
Profile Names=10-year,25-year,50-year,1pct_min,100-year,1pct_plu,500-year
River Rch & RM= Stream0804,Reach-1,23442
     418     663     880     567    1132    2258    1853
River Rch & RM= Stream0804,Reach-1,20202
     763    1255    1708    1126    2246    4482    3851
River Rch & RM= Stream0804,Reach-1,18385
    1136    1905    2626    1751    3494    6971    6131
River Rch & RM= Stream0804,Reach-1,16102
    1202    2018    2783    1856    3703    7388    6498
River Rch & RM= Stream0804,Reach-1,13286
    1763    3003    4181    2809    5605   11183    9994
River Rch & RM= Stream0804,Reach-1,6976
    1942    3310    4611    3097    6180   12331   11016
Boundary for River Rch & Prof#=Stream0804,Reach-1,1
Up Type=0
Dn Type=3
Dn Slope=0.005
Boundary for River Rch & Prof#=Stream0804,Reach-1,2
Up Type=0
Dn Type=3
Dn Slope=0.005
Boundary for River Rch & Prof#=Stream0804,Reach-1,3
Up Type=0
Dn Type=3
Dn Slope=0.005
Boundary for River Rch & Prof#=Stream0804,Reach-1,4
Up Type=0
Dn Type=3
Dn Slope=0.005
Boundary for River Rch & Prof#=Stream0804,Reach-1,5
Up Type=0
Dn Type=3
Dn Slope=0.005
Boundary for River Rch & Prof#=Stream0804,Reach-1,6
Up Type=0
Dn Type=3
Dn Slope=0.005
Boundary for River Rch & Prof#=Stream0804,Reach-1,7
Up Type=0
Dn Type=3
Dn Slope=0.005

--- Stream0804.g01 (geometry) ---

Geom Title=Existing Conditions

River Reach=Stream0804,Reach-1
Reach XY= 30
      2450375.00     13572875.00      2450030.46     13573222.55
      2450071.54     13573573.50      2449777.06     13573930.85
      2449824.67     13575459.97      2449624.56     13575709.82
      2449778.55     13576623.53      2450425.00     13577125.00
      2450573.81     13577685.50      2450227.06     13578330.85
      2450124.60     13579150.00      2450275.24     13579499.92
      2450225.00     13581725.00      2450475.41     13581995.13
      2450282.79     13582271.58      2450224.95     13583555.02
      2450967.67     13584374.90      2450671.24     13585723.44
      2450075.52     13586340.22      2450721.26     13587376.56
      2450583.95     13587781.69      2450875.39     13587995.37
      2450672.00     13588817.05      2450278.75     13589076.55
      2450275.26     13589504.72      2450630.18     13590269.56
      2451280.94     13590672.75      2452016.89     13590677.51
      2452080.34     13591277.74      2452375.00     13591375.00

Type RM Length L Ch R = 1,23442,425,425,425
BEGIN DESCRIPTION:
XS7751
END DESCRIPTION:
XS GIS Cut Line= 2
      2450040.07     13572673.34      2450719.41     13573129.00
#Sta/Elev= 30
  4613.7  353.80  4655.6  352.30  4667.8  353.03  4676.7  352.69  4718.7  349.52
  4748.7  350.33  4769.7  348.31  4805.7  346.86  4820.7  346.54  4841.7  347.45
  4884.5  344.69  4913.8  345.40  4928.8  344.15  4954.8  343.86  4955.0  343.36
  4958.5  343.36  4958.8  343.86  4992.9  343.89  5015.8  345.57  5042.8  344.88
  5087.8  345.81  5101.3  345.38  5209.7  349.84  5231.9  351.24  5267.9  351.81
  5318.0  353.67  5345.9  355.61  5354.1  354.96  5367.0  355.90  5431.7  357.50
#Mann=3,-1,0
  4613.7    0.05       0  4954.8    0.05       0  4958.8    0.05       0
Bank Sta=4954.8,4958.8
Exp/Cntr=0.3,0.1

Type RM Length L Ch R = 1,23017,431,431,431
BEGIN DESCRIPTION:
Stream0804 50.0
END DESCRIPTION:
XS GIS Cut Line= 3
      2449874.99     13572924.99      2450075.00     13573175.00
      2450674.98     13573374.99
#Sta/Elev= 30
  4680.1  351.06  4708.1  348.75  4736.9  349.33  4772.2  346.46  4801.0  347.08
  4836.2  343.89  4885.8  343.96  4900.2  342.85  4936.2  341.55  4972.3  340.66
  4986.6  340.77  4995.1  340.57  4995.3  340.07  4998.8  340.07  4999.1  340.57
  5031.9  340.74  5053.0  341.65  5095.1  342.14  5116.2  343.26  5137.3  343.01
  5141.7  343.33  5168.9  344.90  5263.8  347.34  5284.9  348.62  5348.1  349.75
  5400.8  352.41  5485.2  355.67  5537.9  358.22  5569.5  358.38  5632.7  359.68
#Mann=5,-1,0
  4680.1    0.05       0  4986.6   0.035       0  4995.1   0.035       0
  4999.1   0.035       0  5141.7    0.05       0
Bank Sta=4995.1,4999.1
Exp/Cntr=0.3,0.1

Type RM Length L Ch R = 1,22586,470,470,470
BEGIN DESCRIPTION:
Stream0804 49.0
END DESCRIPTION:
XS GIS Cut Line= 3
      2449674.99     13573024.98      2450075.00     13573575.00
      2450375.00     13573575.00
#Sta/Elev= 30
  4324.5  351.45  4411.1  352.29  4417.6  352.12  4423.8  349.45  4434.8  349.32
  4458.0  348.60  4583.0  346.93  4658.3  343.74  4689.7  342.47  4723.2  338.02
  4723.5  337.52  4727.2  338.02  4754.6  339.78  4760.8  338.21  4769.3  340.82
  4775.5  338.35  4790.1  344.25  4796.3  343.06  4804.8  345.12  4811.0  343.93
  4819.1  346.59  4846.6  347.28  4855.1  345.69  4861.2  346.93  4875.9  341.04
  4882.1  342.90  4890.6  339.79  4961.7  338.27  5104.6  340.23  5304.6  347.52
#Mann=6,-1,0
  4324.5   0.035       0  4434.8    0.05       0  4458.0   0.035       0
  4658.3    0.05       0  4723.2    0.05       0  4727.2    0.05       0
Bank Sta=4723.2,4727.2
Exp/Cntr=0.3,0.1

Type RM Length L Ch R = 1,22116,499,499,499
BEGIN DESCRIPTION:
Stream0804 48.0
END DESCRIPTION:
XS GIS Cut Line= 3
      2449175.03     13573875.00      2449775.00     13573925.00
      2450375.00     13574125.00
#Sta/Elev= 30
  4394.1  343.52  4443.1  342.85  4504.4  340.60  4604.8  339.24  4644.9  337.76
  4692.6  338.24  4734.8  337.86  4823.2  336.83  4855.7  336.67  4944.0  333.25
  4944.2  332.75  4947.7  332.75  4948.0  333.25  4956.0  333.98  4986.1  334.23
  5069.9  333.37  5112.1  334.65  5143.0  334.78  5175.3  336.17  5207.0  334.13
  5217.5  335.54  5245.7  335.96  5333.5  338.09  5407.2  339.12  5417.8  339.77
  5431.4  341.61  5449.4  344.45  5459.9  347.10  5470.5  348.19  5628.6  349.67
#Mann=9,-1,0
  4394.1    0.05       0  4443.1    0.07       0  4734.8    0.05       0
  4823.2    0.07       0  4944.0    0.07       0  4948.0    0.07       0
  5143.0   0.035       0  5245.7    0.05       0  5431.4   0.035       0
Bank Sta=4944,4948
Exp/Cntr=0.3,0.1

Type RM Length L Ch R = 1,21617,466,466,466
BEGIN DESCRIPTION:
Stream0804 47.0
END DESCRIPTION:
XS GIS Cut Line= 3
      2449325.04     13574275.01      2449775.00     13574425.00
      2450324.98     13574325.00
#Sta/Elev= 30
  4526.1  342.26  4768.5  334.72  4831.7  334.31  4860.8  332.39  4937.2  329.55
  5002.9  329.38  5018.7  328.46  5019.0  327.96  5022.7  328.46  5051.2  329.54
  5102.0  329.37  5112.2  330.50  5144.0  331.36  5173.2  334.65  5192.2  336.01
  5197.3  335.54  5213.8  337.44  5230.0  336.82  5244.3  335.85  5274.8  336.26
  5291.8  339.43  5304.0  340.40  5346.0  340.00  5420.9  342.09  5457.8  344.69
  5467.9  346.60  5475.0  349.11  5499.1  348.38  5508.6  349.13  5559.4  349.21
#Mann=8,-1,0
  4526.1    0.07       0  4860.8    0.05       0  5018.7    0.05       0
  5022.7    0.05       0  5230.0   0.035       0  5291.8    0.05       0
  5475.0   0.035       0  5499.1    0.05       0
Bank Sta=5018.7,5022.7
Exp/Cntr=0.3,0.1

Type RM Length L Ch R = 1,21151,500,500,500
BEGIN DESCRIPTION:
Stream0804 46.0
END DESCRIPTION:
XS GIS Cut Line= 3
      2449275.04     13574425.03      2449825.00     13574875.00
      2450425.00     13574475.00
#Sta/Elev= 30
  4289.4  340.54  4459.3  336.83  4629.8  336.39  4665.3  334.87  4729.4  333.69
  4758.1  332.61  4772.4  330.93  4910.9  328.10  4992.8  324.43  4994.8  320.50
  4995.0  320.00  4998.8  320.50  5003.0  320.50  5007.5  323.90  5032.4  326.12
  5049.6  327.63  5130.7  327.16  5283.6  330.76  5288.4  331.70  5295.9  331.12
  5311.0  332.48  5338.5  332.75  5353.0  333.21  5368.1  335.23  5404.1  335.22
  5488.2  338.81  5599.4  342.92  5649.0  346.63  5698.6  347.84  5721.1  349.68
#Mann=11,-1,0
  4289.4    0.07       0  4459.3    0.05       0  4629.8   0.035       0
  4665.3    0.05       0  4910.9    0.16       0  4994.8    0.07       0
  4998.8    0.16       0  5032.4    0.05       0  5283.6   0.035       0
  5338.5    0.05       0  5488.2   0.035       0
Bank Sta=4994.8,4998.8
Exp/Cntr=0.3,0.1

Type RM Length L Ch R = 1,20651,449,449,449
BEGIN DESCRIPTION:
Stream0804 45.0
END DESCRIPTION:
XS GIS Cut Line= 3
      2449475.01     13574975.02      2449825.00     13575375.00
      2450025.01     13575475.00
#Sta/Elev= 30
  4468.4  329.22  4638.4  326.48  4653.0  326.09  4667.2  326.30  4673.9  325.81
  4694.7  325.51  4766.4  324.88  4843.8  323.42  4872.2  323.62  4900.7  322.46
  4929.2  322.46  4933.7  322.81  4950.1  324.06  4961.9  323.88  4986.1  323.03
  4996.6  322.15  5008.3  321.74  5022.2  321.85  5030.0  321.25  5044.6  320.75
  5065.0  317.56  5065.2  317.06  5068.7  317.06  5069.0  317.56  5075.4  321.04
  5080.9  321.95  5097.7  325.88  5120.1  326.26  5209.5  330.23  5223.5  330.43
#Mann=7,-1,0
  4468.4    0.07       0  4638.4    0.16       0  4766.4    0.07       0
  4933.7    0.16       0  5030.0    0.07       0  5065.0    0.07       0
  5069.0    0.07       0
Bank Sta=5065,5069
Exp/Cntr=0.3,0.1

Type RM Length L Ch R = 1,20202,452,452,452
BEGIN DESCRIPTION:
Stream0804 44.0
END DESCRIPTION:
XS GIS Cut Line= 3
      2449324.99     13576025.01      2449625.00     13575725.00
      2449825.02     13575725.00
#Sta/Elev= 30
  4576.3  327.84  4592.0  327.39  4604.6  327.07  4618.7  326.30  4632.9  326.58
  4675.3  325.07  4731.9  323.67  4774.3  324.53  4802.6  323.80  4816.7  323.02
  4830.9  322.58  4845.0  321.59  4873.3  323.15  4901.6  323.72  4929.9  323.06
  4944.0  323.27  4958.2  322.64  4997.0  317.53  5003.1  317.53  5008.6  316.79
  5008.8  316.29  5012.3  316.29  5012.6  316.79  5030.6  318.27  5040.6  318.47
  5060.6  320.89  5130.6  324.40  5150.6  325.97  5170.6  326.69  5200.6  326.95
#Mann=4,-1,0
  4576.3   0.035       0  4592.0    0.07       0  5008.6    0.07       0
  5012.6    0.07       0
Bank Sta=5008.6,5012.6
Exp/Cntr=0.3,0.1

Type RM Length L Ch R = 1,19750,499,499,499
BEGIN DESCRIPTION:
Stream0804 43.0
END DESCRIPTION:
XS GIS Cut Line= 4
      2449106.64     13576256.64      2449551.79     13576214.28
      2449775.00     13576125.00      2449975.02     13576024.99
#Sta/Elev= 30
  4312.0  337.60  4440.9  332.33  4451.0  332.47  4486.9  330.14  4491.9  330.49
  4511.3  329.32  4521.3  329.47  4639.9  324.71  4682.0  322.93  4762.9  321.38
  4841.9  320.74  4870.0  320.47  4977.2  319.66  4990.1  319.26  5008.0  317.20
  5013.5  317.51  5044.3  315.82  5050.7  314.31  5050.9  313.81  5054.4  313.81
  5054.7  314.31  5058.3  315.09  5066.7  318.97  5080.6  320.74  5097.4  320.38
  5147.7  323.38  5156.1  324.52  5196.8  326.44  5214.8  326.86  5223.2  327.65
#Mann=9,-1,0
  4312.0    0.07       0  4639.9    0.12       0  4762.9    0.07       0
  4841.9    0.12       0  4870.0    0.07       0  4977.2    0.12       0
  5050.7    0.05       0  5054.7    0.12       0  5196.8    0.07       0
Bank Sta=5050.7,5054.7
Exp/Cntr=0.3,0.1

Type RM Length L Ch R = 1,19251,441,441,441
BEGIN DESCRIPTION:
Stream0804 42.0
END DESCRIPTION:
XS GIS Cut Line= 3
      2449375.00     13577025.00      2449775.00     13576625.00
      2450024.98     13576475.01
#Sta/Elev= 30
  4430.4  339.19  4458.7  338.17  4487.0  335.72  4586.0  330.01  4600.1  328.50
  4614.2  328.53  4642.5  326.19  4674.8  324.61  4727.4  322.83  4741.5  321.72
  4755.7  322.08  4769.8  320.90  4779.7  320.87  4802.2  319.84  4911.2  319.28
  4939.5  316.93  4999.0  314.48  5003.9  308.25  5007.6  308.14  5007.9  307.64
  5011.5  307.64  5011.7  308.14  5019.4  311.89  5031.1  313.18  5040.8  312.93
  5062.2  316.04  5068.0  316.31  5077.7  318.16  5188.2  321.72  5287.6  326.07
#Mann=7,-1,0
  4430.4    0.07       0  4674.8    0.16       0  4779.7    0.07       0
  4802.2    0.16       0  5007.6    0.07       0  5011.7    0.16       0
  5188.2    0.07       0
Bank Sta=5007.6,5011.7
Exp/Cntr=0.3,0.1

Type RM Length L Ch R = 1,18810,425,425,425
BEGIN DESCRIPTION:
Stream0804 41.0
END DESCRIPTION:
XS GIS Cut Line= 3
      2449375.02     13577624.98      2450075.00     13576925.00
      2450125.00     13576525.04
#Sta/Elev= 30
  4005.7  350.21  4009.2  350.21  4019.8  352.99  4048.1  355.37  4062.2  354.60
  4076.4  351.60  4090.5  351.01  4104.7  349.11  4118.8  344.54  4133.0  342.77
  4260.2  337.62  4316.8  333.97  4606.7  321.79  4712.8  316.35  4769.3  314.48
  4854.5  314.88  4910.8  315.40  4939.1  314.59  4967.3  307.81  4979.4  306.62
  4979.7  306.12  4983.5  306.62  4992.1  310.28  5038.5  311.05  5076.2  315.34
  5106.5  316.19  5141.5  315.83  5354.9  324.31  5398.6  325.84  5398.7  325.84
#Mann=7,-1,0
  4005.7    0.07       0  4854.5    0.16       0  4979.4    0.07       0
  4983.5    0.16       0  5141.5    0.07       0  5354.9   0.035       0
  5398.6    0.07       0
Bank Sta=4979.4,4983.5
Exp/Cntr=0.3,0.1

Type RM Length L Ch R = 1,18385,483,483,483
BEGIN DESCRIPTION:
Stream0804 40.0
END DESCRIPTION:
XS GIS Cut Line= 3
      2449625.02     13577674.99      2450425.00     13577125.00
      2450824.99     13577175.00
#Sta/Elev= 30
  4029.2  339.45  4178.3  332.84  4502.7  319.25  4805.8  312.91  4819.3  310.66
  4828.2  307.62  4834.2  308.08  4842.2  306.18  4864.0  306.98  4870.1  305.87
  4878.6  306.74  4885.0  310.09  4920.8  309.39  4935.7  311.93  4941.8  309.53
  4963.6  305.80  4968.8  298.75  4969.2  298.25  4974.4  298.75  4992.6  300.08
  4997.0  305.72  5010.1  304.97  5037.8  312.19  5042.8  311.66  5088.1  316.77
  5186.9  319.50  5204.1  318.80  5231.8  323.31  5285.7  325.75  5403.1  333.07
#Mann=7,-1,0
  4029.2    0.07       0  4178.3    0.16       0  4968.8    0.07       0
  4974.4    0.16       0  5088.1    0.07       0  5186.9   0.035       0
  5285.7    0.07       0
Bank Sta=4968.8,4974.4
Exp/Cntr=0.3,0.1

Type RM Length L Ch R = 1,17902,446,446,446
BEGIN DESCRIPTION:
Stream0804 39.0
END DESCRIPTION:
XS GIS Cut Line= 3
      2449725.05     13577724.99      2450525.00     13577575.00
      2450725.00     13577475.00
#Sta/Elev= 30
  4190.8  334.81  4220.8  333.46  4302.7  328.56  4404.4  325.06  4542.6  318.66
  4607.9  317.22  4677.2  314.33  4810.5  310.95  4878.4  311.12  4925.8  311.32
  4939.3  310.62  4953.8  308.80  4964.0  305.81  4979.0  303.15  4984.3  301.05
  4991.7  296.46  4992.2  295.96  4997.3  296.46  5002.2  298.42  5007.5  298.42
  5018.7  304.41  5057.8  311.25  5087.8  313.10  5130.5  315.90  5147.2  319.50
  5161.2  320.63  5183.8  320.20  5192.0  318.22  5199.3  318.61  5228.3  322.11
#Mann=11,-1,0
  4190.8    0.07       0  4220.8    0.16       0  4677.2    0.07       0
  4878.4    0.12       0  4939.3    0.16       0  4979.0    0.12       0
  4991.7    0.07       0  4997.3    0.12       0  5087.8    0.07       0
  5183.8   0.035       0  5199.3    0.07       0
Bank Sta=4991.7,4997.3
Exp/Cntr=0.3,0.1

Type RM Length L Ch R = 1,17456,443,443,443
BEGIN DESCRIPTION:
Stream0804 38.0
END DESCRIPTION:
XS GIS Cut Line= 3
      2450225.00     13577875.00      2450475.00     13577975.00
      2450725.04     13577975.00
#Sta/Elev= 30
  4725.7  312.64  4779.6  310.29  4818.6  309.72  4833.4  309.93  4865.7  309.62
  4872.5  309.26  4877.8  309.50  4955.9  309.13  4973.4  305.05  4980.2  303.74
  4985.5  303.37  4992.3  301.37  4997.5  301.37  5002.2  295.52  5002.6  295.02
  5007.3  295.02  5007.8  295.52  5015.0  297.88  5025.0  298.66  5035.0  302.43
  5045.0  304.76  5055.0  306.28  5065.0  309.84  5075.0  311.28  5115.0  312.56
  5155.0  315.45  5175.0  315.40  5185.0  316.27  5205.1  317.03  5245.0  319.14
#Mann=4,-1,0
  4725.7    0.12       0  5002.2    0.07       0  5007.8    0.12       0
  5205.1   0.035       0
Bank Sta=5002.2,5007.8
Exp/Cntr=0.3,0.1

Type RM Length L Ch R = 1,17013,429,429,429
BEGIN DESCRIPTION:
Stream0804 37.0
END DESCRIPTION:
XS GIS Cut Line= 3
      2450074.97     13578325.00      2450225.00     13578325.00
      2451025.01     13578075.00
#Sta/Elev= 30
  4844.7  316.73  4904.7  312.60  4940.6  306.64  4974.7  302.24  5011.0  294.97
  5016.2  297.25  5023.3  294.72  5023.8  294.22  5029.0  294.72  5043.5  299.75
  5048.7  297.30  5075.9  303.27  5081.2  301.64  5108.4  306.83  5113.6  305.88
  5130.9  308.17  5158.7  308.70  5163.3  308.78  5262.7  308.23  5366.7  310.98
  5470.6  316.29  5539.5  319.66  5546.3  321.00  5574.6  319.97  5591.9  321.04
  5616.5  319.77  5643.8  325.41  5678.6  326.99  5791.0  333.23  5832.9  334.27
#Mann=11,-1,0
  4844.7    0.16       0  4940.6    0.12       0  5023.3    0.07       0
  5029.0    0.12       0  5158.7    0.07       0  5163.3    0.12       0
  5262.7    0.16       0  5366.7    0.12       0  5470.6    0.16       0
  5574.6   0.035       0  5678.6    0.07       0
Bank Sta=5023.3,5029
Exp/Cntr=0.3,0.1

Type RM Length L Ch R = 1,16584,482,482,482
BEGIN DESCRIPTION:
Stream0804 36.0
END DESCRIPTION:
XS GIS Cut Line= 3
      2450025.05     13578675.01      2450225.00     13578725.00
      2450624.99     13578725.00
#Sta/Elev= 30
  4798.5  316.00  4808.8  315.28  4829.4  314.71  4839.7  313.51  4850.0  313.43
  4857.7  312.67  4899.0  310.38  4922.1  308.72  4927.3  306.91  4932.5  305.09
  4940.2  303.32  4945.3  303.21  4963.4  299.85  4981.4  297.88  4986.6  296.90
  4991.4  290.65  4991.9  290.15  4996.7  290.15  4997.1  290.65  5007.1  290.79
  5014.6  294.42  5024.6  300.99  5044.6  306.05  5049.9  306.22  5074.6  306.69
  5148.3  305.45  5274.6  307.02  5324.6  308.04  5364.6  308.13  5404.6  309.00
#Mann=6,-1,0
  4798.5    0.16       0  4927.3    0.12       0  4991.4    0.07       0
  4997.1    0.12       0  5049.9    0.07       0  5148.3    0.05       0
Bank Sta=4991.4,4997.1
Exp/Cntr=0.3,0.1

Type RM Length L Ch R = 1,16102,448,448,448
BEGIN DESCRIPTION:
Stream0804 35.0
END DESCRIPTION:
XS GIS Cut Line= 3
      2449924.99     13579024.99      2450125.00     13579175.00
      2450474.97     13578975.02
#Sta/Elev= 30
  4751.0  312.06  4793.7  311.66  4872.9  307.74  4879.1  306.11  4893.7  304.53
  4943.7  301.12  4993.7  296.69  4997.9  291.59  5003.9  291.59  5006.0  288.47
  5006.5  287.97  5011.9  288.47  5014.7  289.29  5024.1  289.37  5030.5  296.18
  5036.3  294.71  5046.4  297.64  5052.1  296.77  5068.0  300.98  5073.7  301.39
  5081.6  303.47  5111.2  305.08  5162.6  304.24  5235.0  303.59  5250.8  302.25
  5256.6  302.81  5272.4  301.31  5315.6  302.47  5331.4  304.42  5404.1  305.39
#Mann=4,-1,0
  4751.0    0.16       0  5006.0    0.07       0  5011.9    0.16       0
  5162.6    0.05       0
Bank Sta=5006,5011.9
Exp/Cntr=0.3,0.1

Type RM Length L Ch R = 1,15654,482,482,482
BEGIN DESCRIPTION:
Stream0804 34.0
END DESCRIPTION:
XS GIS Cut Line= 3
      2450024.97     13579575.00      2450275.00     13579575.00
      2450524.97     13579575.00
#Sta/Elev= 30
  4749.5  308.57  4755.3  308.35  4789.5  306.41  4839.5  304.20  4879.5  302.68
  4889.5  302.78  4899.5  302.38  4929.5  296.23  4939.5  295.28  4959.5  294.92
  4969.5  293.03  4986.4  287.06  4986.9  286.56  4992.1  286.56  4992.6  287.06
  4997.0  288.81  5002.0  288.81  5009.5  294.47  5013.2  295.77  5019.5  297.99
  5039.5  298.46  5049.5  299.52  5059.5  301.03  5071.6  302.01  5089.5  303.45
  5099.5  303.44  5139.5  305.16  5169.5  305.76  5239.5  308.52  5249.5  308.65
#Mann=6,-1,0
  4749.5    0.07       0  4755.3    0.16       0  4986.4    0.07       0
  4992.6    0.16       0  5013.2    0.07       0  5071.6    0.05       0
Bank Sta=4986.4,4992.6
Exp/Cntr=0.3,0.1

Type RM Length L Ch R = 1,15172,440,440,440
BEGIN DESCRIPTION:
Stream0804 33.0
END DESCRIPTION:
XS GIS Cut Line= 3
      2449974.99     13579975.00      2450175.00     13580025.00
      2450575.03     13579924.99
#Sta/Elev= 30
  4789.5  312.69  4944.1  306.17  4964.7  304.31  4972.5  300.62  4977.6  300.57
  4985.4  296.49  4993.1  288.04  4998.2  288.04  5002.9  285.54  5003.4  285.04
  5009.1  285.54  5018.9  286.36  5026.6  289.97  5036.9  292.88  5047.2  294.25
  5054.9  296.39  5060.1  296.03  5067.8  298.49  5088.4  298.26  5119.4  299.76
  5137.4  299.48  5178.6  300.49  5302.3  304.94  5335.8  306.86  5343.6  307.97
  5348.7  307.55  5377.1  310.71  5384.8  310.82  5389.9  309.75  5408.0  310.71
#Mann=3,-1,0
  4789.5    0.07       0  5002.9    0.07       0  5009.1    0.07       0
Bank Sta=5002.9,5009.1
Exp/Cntr=0.3,0.1

Type RM Length L Ch R = 1,14732,467,467,467
BEGIN DESCRIPTION:
Stream0804 32.0
END DESCRIPTION:
XS GIS Cut Line= 3
      2450025.00     13580425.00      2450225.00     13580425.00
      2450525.04     13580224.98
#Sta/Elev= 30
  4800.0  308.68  4830.0  307.15  4860.0  306.51  4893.3  304.70  4900.0  303.93
  4950.0  294.22  4960.0  291.36  4970.0  290.32  4980.0  290.37  4990.0  289.22
  4997.5  287.51  5003.0  287.51  5007.5  285.12  5019.4  284.13  5019.9  283.63
  5025.2  283.63  5025.7  284.13  5028.5  284.18  5036.1  287.24  5043.6  292.51
  5049.6  290.92  5058.6  295.82  5085.6  296.08  5097.1  295.66  5121.7  295.76
  5151.7  297.38  5223.8  299.82  5252.4  300.37  5317.0  304.02  5360.6  305.20
#Mann=5,-1,0
  4800.0    0.07       0  4893.3    0.16       0  5019.4    0.07       0
  5025.7    0.16       0  5097.1    0.07       0
Bank Sta=5019.4,5025.7
Exp/Cntr=0.3,0.1

Type RM Length L Ch R = 1,14265,432,432,432
BEGIN DESCRIPTION:
Stream0804 31.0
END DESCRIPTION:
XS GIS Cut Line= 3
      2450025.01     13580825.00      2450275.00     13580875.00
      2450474.96     13580875.00
#Sta/Elev= 30
  4740.2  305.31  4770.8  303.84  4811.6  302.74  4862.6  298.79  4893.2  297.46
  4903.4  296.74  4913.6  295.51  4923.8  293.27  4944.1  289.53  4954.3  288.15
  4964.5  287.39  4974.7  287.02  4984.9  284.74  4989.3  282.83  4989.8  282.33
  4995.3  282.33  4995.8  282.83  5005.1  282.91  5015.1  284.25  5025.1  286.68
  5035.1  288.14  5045.1  289.29  5055.1  290.90  5065.1  294.02  5075.1  295.55
  5085.1  298.09  5115.1  299.89  5145.1  300.89  5155.1  301.66  5195.1  303.52
#Mann=3,-1,0
  4740.2    0.07       0  4989.3    0.07       0  4995.8    0.07       0
Bank Sta=4989.3,4995.8
Exp/Cntr=0.3,0.1

Type RM Length L Ch R = 1,13833,295,295,295
BEGIN DESCRIPTION:
Stream0804 30.0
END DESCRIPTION:
XS GIS Cut Line= 3
      2449975.05     13581125.02      2450225.00     13581225.00
      2450425.03     13581174.99
#Sta/Elev= 30
  4730.7  298.03  4740.1  297.87  4752.2  296.87  4806.0  295.69  4853.2  295.45
  4859.9  294.83  4870.7  292.84  4892.2  287.95  4901.6  287.31  4907.0  287.83
  4931.2  283.93  4936.6  285.76  4955.5  281.30  4960.9  281.39  4964.3  280.53
  4964.8  280.03  4970.3  280.03  4970.8  280.53  4978.4  281.04  4985.1  285.61
  4990.5  284.24  4997.2  289.84  5002.5  289.84  5010.2  292.48  5017.9  294.46
  5041.1  294.69  5082.4  296.79  5092.7  296.61  5182.9  301.33  5206.1  302.01
#Mann=3,-1,0
  4730.7    0.07       0  4964.3    0.07       0  4970.8    0.07       0
Bank Sta=4964.3,4970.8
Exp/Cntr=0.3,0.1

Type RM Length L Ch R = 1,13538,252,252,252
BEGIN DESCRIPTION:
H21082
END DESCRIPTION:
XS GIS Cut Line= 3
      2449862.99     13581145.02      2450145.27     13581510.33
      2450551.05     13581564.16
#Sta/Elev= 30
  4457.9  298.56  4502.1  297.32  4516.6  296.00  4677.8  293.96  4817.5  293.28
  4873.4  292.88  4879.7  287.18  4887.6  287.88  4894.2  292.21  4908.7  292.98
  4921.9  292.07  4939.5  286.56  4959.6  284.37  4961.7  283.45  4971.3  279.79
  4976.5  279.29  4977.0  278.79  4983.1  279.29  4989.0  282.76  4994.0  283.54
  5000.0  283.22  5010.1  285.13  5020.2  289.56  5030.3  291.87  5040.3  293.03
  5090.8  292.21  5121.0  292.86  5292.4  302.19  5297.4  301.67  5328.9  303.47
#Mann=7,-1,0
  4457.9    0.07       0  4677.8    0.16       0  4817.5    0.07       0
  4961.7    0.16       0  4971.3    0.07       0  4976.5    0.07       0
  4983.1    0.07       0
Bank Sta=4976.5,4983.1
Exp/Cntr=0.3,0.1

Type RM Length L Ch R = 1,13286,421,421,421
BEGIN DESCRIPTION:
Stream0804 29.0
END DESCRIPTION:
XS GIS Cut Line= 3
      2449725.98     13581979.40      2450232.44     13581771.84
      2450525.02     13581624.99
#Sta/Elev= 30
  4423.3  313.17  4448.7  312.35  4472.7  310.00  4590.1  302.44  4692.4  295.47
  4757.3  292.84  4769.0  290.20  4787.6  288.75  4841.0  281.00  4854.5  281.55
  4870.4  288.32  4876.1  287.96  4899.8  290.02  4918.4  289.88  4923.8  288.27
  4947.8  287.62  4953.2  284.77  4962.6  285.60  4976.9  283.27  4993.7  282.69
  5011.4  277.12  5011.9  276.62  5020.5  277.12  5038.3  278.79  5043.9  285.57
  5051.8  288.51  5074.2  291.28  5163.7  293.21  5253.2  297.36  5298.0  300.63
#Mann=4,-1,0
  4423.3    0.16       0  4590.1    0.07       0  5011.4    0.07       0
  5020.5    0.07       0
Bank Sta=5011.4,5020.5
Exp/Cntr=0.3,0.1

Type RM Length L Ch R = 1,12865,419,419,419
BEGIN DESCRIPTION:
Stream0804 28.0
END DESCRIPTION:
XS GIS Cut Line= 3
      2450025.00     13582125.00      2450425.00     13582075.00
      2450625.03     13582125.01
#Sta/Elev= 30
  4592.2  293.80  4647.1  291.36  4733.3  287.35  4770.1  282.26  4783.7  278.19
  4796.3  277.41  4803.8  281.69  4813.9  282.67  4834.1  282.55  4871.9  286.47
  4904.6  287.83  4914.7  287.26  4934.8  284.03  4965.1  284.37  4975.2  282.58
  4985.2  277.31  4992.8  276.39  5005.6  277.07  5013.4  276.43  5018.5  277.62
  5021.7  276.11  5022.2  275.61  5030.8  276.11  5054.6  280.59  5059.7  285.53
  5067.5  287.06  5095.8  291.28  5137.0  294.89  5141.7  294.47  5201.5  296.05
#Mann=6,-1,0
  4592.2    0.16       0  4647.1    0.07       0  4770.1    0.12       0
  5021.7    0.07       0  5030.8    0.12       0  5141.7    0.07       0
Bank Sta=5021.7,5030.8
Exp/Cntr=0.3,0.1

Type RM Length L Ch R = 1,12446,469,469,469
BEGIN DESCRIPTION:
Stream0804 27.0
END DESCRIPTION:
XS GIS Cut Line= 3
      2450074.96     13582374.99      2450325.00     13582425.00
      2450574.96     13582275.02
#Sta/Elev= 30
  4744.9  293.41  4846.9  287.32  4887.7  284.37  4918.3  282.73  4928.5  283.08
  4935.5  282.26  4944.6  281.73  4959.1  281.35  4969.3  280.41  4985.1  273.51
  4985.6  273.01  4993.8  273.01  4994.3  273.51  4997.3  277.24  5002.8  277.24
  5007.7  282.11  5013.5  281.84  5023.2  283.55  5034.9  283.70  5044.6  285.08
  5050.4  284.34  5066.0  285.02  5071.8  284.00  5093.2  286.87  5116.5  288.17
  5130.1  288.01  5219.5  291.12  5237.4  291.28  5276.4  292.02  5291.4  292.52
#Mann=7,-1,0
  4744.9    0.16       0  4935.5    0.12       0  4944.6    0.16       0
  4985.1    0.07       0  4994.3    0.16       0  5237.4    0.12       0
  5276.4    0.05       0
Bank Sta=4985.1,4994.3
Exp/Cntr=0.3,0.1

Type RM Length L Ch R = 1,11977,486,486,486
BEGIN DESCRIPTION:
Stream0804 26.0
END DESCRIPTION:
XS GIS Cut Line= 3
      2449975.00     13583025.00      2450375.00     13582875.00
      2450774.99     13582775.00
#Sta/Elev= 30
  4578.0  296.82  4653.7  293.88  4673.2  291.81  4731.2  288.60  4794.3  285.63
  4844.1  282.11  4874.4  281.33  4879.7  282.60  4904.6  279.54  4910.0  279.99
  4929.6  278.68  4973.2  279.15  4983.8  278.49  4990.1  276.92  4995.4  278.87
  5002.5  277.24  5007.1  277.24  5015.5  274.69  5018.3  271.33  5018.8  270.83
  5028.1  271.33  5028.4  271.96  5036.1  272.34  5051.7  277.75  5064.5  281.33
  5098.0  284.89  5284.0  286.73  5317.0  289.02  5358.2  290.11  5417.5  294.42
#Mann=7,-1,0
  4578.0    0.16       0  4731.2    0.12       0  5007.1    0.16       0
  5018.3    0.07       0  5028.1    0.16       0  5051.7    0.12       0
  5284.0    0.07       0
Bank Sta=5018.3,5028.1
Exp/Cntr=0.3,0.1

Type RM Length L Ch R = 1,11491,541,541,541
BEGIN DESCRIPTION:
Stream0804 25.0
END DESCRIPTION:
XS GIS Cut Line= 3
      2450025.03     13583325.00      2450275.00     13583325.00
      2451075.00     13582775.00
#Sta/Elev= 30
  4754.6  294.49  4874.6  285.87  4894.6  281.98  4944.6  276.55  4954.6  273.76
  4959.7  270.48  4960.2  269.98  4969.5  270.48  5012.0  280.62  5033.0  276.86
  5057.2  278.72  5079.6  280.38  5113.5  278.78  5206.2  283.66  5248.1  284.14
  5263.0  282.03  5313.7  284.87  5507.9  285.63  5583.0  290.06  5642.8  293.84
  5717.0  300.47  5758.9  301.63  5781.2  304.53  5809.6  304.61  5839.4  308.46
  5866.5  308.16  5902.6  311.48  5931.3  311.57  5953.1  314.93  5975.4  314.38
#Mann=7,-1,0
  4754.6    0.16       0  4959.7    0.07       0  4969.5    0.16       0
  5057.2    0.07       0  5079.6    0.12       0  5583.0    0.16       0
  5642.8    0.07       0
Bank Sta=4959.7,4969.5
Exp/Cntr=0.3,0.1

Type RM Length L Ch R = 1,10950,357,357,357
BEGIN DESCRIPTION:
Stream0804 24.0
END DESCRIPTION:
XS GIS Cut Line= 3
      2449975.11     13583809.96      2450406.78     13583722.80
      2451202.53     13583399.52
#Sta/Elev= 30
  4508.5  297.32  4752.7  284.40  4783.8  283.19  4851.8  283.66  4875.7  281.44
  4906.3  280.80  4917.0  278.06  4948.9  274.79  4973.5  268.70  4974.0  268.20
  4983.4  268.70  5007.9  275.81  5054.9  280.70  5098.1  280.98  5115.0  279.46
  5120.4  280.89  5150.3  281.15  5162.8  281.25  5168.6  279.59  5173.9  280.90
  5192.6  277.52  5222.1  277.72  5227.6  280.18  5238.4  281.82  5301.2  282.76
  5395.8  285.62  5475.9  287.18  5608.2  297.25  5698.7  300.03  5807.8  300.32
#Mann=9,-1,0
  4508.5    0.07       0  4752.7    0.12       0  4851.8     0.1       0
  4973.5    0.05       0  4983.4     0.1       0  5150.3    0.12       0
  5301.2     0.1       0  5395.8    0.07       0  5608.2    0.12       0
Bank Sta=4973.5,4983.4
Exp/Cntr=0.3,0.1

Type RM Length L Ch R = 1,10593,470,470,470
BEGIN DESCRIPTION:
Stream0804 23.0
END DESCRIPTION:
XS GIS Cut Line= 5
      2449847.88     13584141.03      2450700.12     13583937.44
      2450725.00     13583925.00      2450743.26     13583911.30
      2451323.21     13583649.41
#Sta/Elev= 30
  4100.3  298.64  4374.9  289.68  4604.6  286.05  4693.7  282.26  4846.8  279.49
  4868.4  276.72  4876.5  279.87  4918.6  279.19  4930.1  275.79  4960.7  271.65
  4968.4  266.03  4968.9  265.53  4978.7  266.03  5001.5  273.74  5011.6  274.02
  5025.1  276.92  5050.1  276.23  5062.1  277.78  5078.7  275.28  5084.2  277.09
  5101.8  276.28  5107.3  277.89  5116.8  276.46  5171.2  280.72  5326.4  286.81
  5349.5  289.11  5430.1  293.33  5493.7  297.45  5539.4  302.60  5663.5  310.28
#Mann=8,-1,0
  4100.3    0.07       0  4604.6    0.12       0  4846.8     0.1       0
  4968.4    0.05       0  4978.7     0.1       0  5062.1    0.12       0
  5430.1    0.07       0  5539.4    0.12       0
Bank Sta=4968.4,4978.7
Exp/Cntr=0.3,0.1

Type RM Length L Ch R = 1,10123,466,466,466
BEGIN DESCRIPTION:
Stream0804 22.0
END DESCRIPTION:
XS GIS Cut Line= 4
      2450041.89     13584427.69      2450664.16     13584368.47
      2450925.00     13584325.00      2451274.98     13584325.00
#Sta/Elev= 30
  4110.3  293.32  4422.8  285.00  4485.1  283.70  4504.2  285.60  4595.6  281.18
  4617.2  281.59  4726.2  279.38  4756.5  279.91  4850.3  277.07  4871.3  273.83
  4878.2  274.22  4888.3  277.43  4911.1  278.14  4954.9  271.65  4959.3  271.14
  4966.9  266.82  4974.4  266.55  4974.9  266.05  4984.7  266.55  4997.3  270.62
  5002.3  270.62  5009.8  273.45  5049.8  278.89  5149.1  285.44  5179.8  287.39
  5219.8  292.01  5267.1  293.05  5299.8  297.46  5329.8  298.19  5349.8  302.35
#Mann=8,-1,0
  4110.3    0.07       0  4422.8    0.12       0  4871.3     0.1       0
  4954.9    0.12       0  4974.4    0.05       0  4984.7    0.12       0
  5149.1   0.035       0  5267.1    0.12       0
Bank Sta=4974.4,4984.7
Exp/Cntr=0.3,0.1

Type RM Length L Ch R = 1,9657,417,417,417
BEGIN DESCRIPTION:
Stream0804 21.0
END DESCRIPTION:
XS GIS Cut Line= 3
      2450575.00     13584725.00      2450925.00     13584725.00
      2451075.00     13584725.00
#Sta/Elev= 30
  4649.9  281.98  4659.9  281.78  4764.0  276.93  4789.9  274.68  4799.9  274.82
  4819.9  273.93  4849.9  275.07  4859.9  276.40  4879.9  276.77  4889.9  276.43
  4919.9  271.78  4929.9  271.04  4939.9  271.40  4949.9  269.59  4954.7  266.81
  4955.2  266.31  4964.6  266.31  4965.1  266.81  4969.9  267.43  4979.9  267.75
  4989.9  269.37  4997.4  271.68  5002.4  271.68  5009.9  273.09  5029.9  274.89
  5079.9  281.46  5089.9  282.21  5099.9  283.51  5118.8  285.06  5149.9  286.80
#Mann=5,-1,0
  4649.9    0.16       0  4764.0    0.12       0  4954.7    0.07       0
  4965.1    0.12       0  5118.8   0.035       0
Bank Sta=4954.7,4965.1
Exp/Cntr=0.3,0.1

Type RM Length L Ch R = 1,9240,480,480,480
BEGIN DESCRIPTION:
Stream0804 20.0
END DESCRIPTION:
XS GIS Cut Line= 3
      2450525.01     13585025.00      2450725.00     13585075.00
      2451125.04     13585025.00
#Sta/Elev= 30
  4794.0  288.74  4804.3  287.86  4812.0  288.49  4853.3  284.58  4866.1  284.46
  4876.5  282.95  4894.5  282.10  4907.4  280.22  4928.0  278.81  4935.7  277.60
  4940.9  278.27  4958.9  272.28  4977.0  265.04  4982.1  264.70  4984.5  261.75
  4985.0  261.25  4994.6  261.25  4995.1  261.75  4997.6  263.67  5010.2  263.29
  5037.9  268.66  5043.0  267.64  5131.2  275.62  5181.6  276.66  5224.2  279.20
  5242.0  280.25  5262.2  280.31  5272.3  282.07  5351.6  288.35  5403.3  291.53
#Mann=5,-1,0
  4794.0   0.035       0  4984.5   0.035       0  4995.1   0.035       0
  5224.2    0.16       0  5351.6    0.07       0
Bank Sta=4984.5,4995.1
Exp/Cntr=0.3,0.1

Type RM Length L Ch R = 1,8760,447,447,447
BEGIN DESCRIPTION:
Stream0804 19.0
END DESCRIPTION:
XS GIS Cut Line= 3
      2450474.96     13585424.99      2450725.00     13585525.00
      2451025.00     13585925.00
#Sta/Elev= 30
  4734.8  278.92  4790.3  277.21  4864.1  274.48  4911.2  274.14  4959.7  266.77
  4982.6  259.58  4983.9  258.34  4984.4  257.84  4994.6  258.34  4994.7  259.33
  5001.4  263.67  5011.4  263.90  5017.6  266.04  5061.4  271.94  5095.8  273.60
  5182.2  275.53  5204.1  273.86  5217.6  271.46  5226.0  267.10  5232.2  269.43
  5233.7  268.86  5240.6  266.21  5246.8  269.64  5254.1  271.29  5317.6  279.48
  5385.6  281.65  5417.6  285.20  5446.8  285.20  5476.0  288.81  5504.1  288.40
#Mann=7,-1,0
  4734.8    0.07       0  4790.3    0.16       0  4983.9    0.07       0
  4994.6    0.16       0  5095.8    0.12       0  5233.7    0.07       0
  5385.6    0.05       0
Bank Sta=4983.9,4994.6
Exp/Cntr=0.3,0.1

Type RM Length L Ch R = 1,8313,453,453,453
BEGIN DESCRIPTION:
Stream0804 18.0
END DESCRIPTION:
XS GIS Cut Line= 3
      2450374.97     13585774.97      2450575.00     13585925.00
      2450775.01     13586125.01
#Sta/Elev= 30
  4754.3  273.48  4817.9  272.82  4826.2  272.95  4832.5  274.21  4854.3  272.18
  4890.8  271.96  4911.6  270.79  4917.9  269.61  4926.2  270.04  4940.8  269.13
  4947.1  267.77  4961.6  267.72  4982.5  265.48  4990.8  263.92  4997.1  260.46
  5001.2  256.73  5012.9  256.19  5013.4  255.69  5024.1  256.19  5046.8  274.29
  5057.3  276.05  5089.2  280.78  5131.6  281.27  5174.0  286.31  5181.1  285.25
  5202.3  285.26  5230.6  288.93  5260.0  288.65  5273.0  288.62  5287.2  289.70
#Mann=5,-1,0
  4754.3    0.16       0  5012.9    0.07       0  5024.1    0.16       0
  5057.3    0.05       0  5260.0   0.035       0
Bank Sta=5012.9,5024.1
Exp/Cntr=0.3,0.1

Type RM Length L Ch R = 1,7860,434,434,434
BEGIN DESCRIPTION:
Stream0804 17.0
END DESCRIPTION:
XS GIS Cut Line= 3
      2449974.98     13586025.00      2450175.00     13586075.00
      2450525.01     13586275.01
#Sta/Elev= 30
  4794.4  279.03  4885.1  273.04  4907.8  271.71  4918.1  269.11  4936.1  260.80
  4943.4  255.85  4943.9  255.35  4954.2  255.35  4954.7  255.85  4982.5  256.57
  4983.9  257.21  4990.3  260.13  4998.0  261.54  5014.2  262.79  5035.8  262.72
  5093.5  267.53  5104.2  268.62  5110.7  270.15  5175.5  272.11  5212.9  274.22
  5228.8  276.27  5242.4  277.15  5277.7  277.60  5300.0  281.21  5316.5  281.95
  5323.1  281.39  5346.1  281.75  5352.6  282.94  5395.8  286.33  5403.7  285.28
#Mann=7,-1,0
  4794.4    0.16       0  4885.1    0.07       0  4943.4    0.07       0
  4954.7    0.07       0  4983.9    0.12       0  5093.5   0.035       0
  5316.5    0.05       0
Bank Sta=4943.4,4954.7
Exp/Cntr=0.3,0.1

Type RM Length L Ch R = 1,7426,450,450,450
BEGIN DESCRIPTION:
Stream0804 16.0
END DESCRIPTION:
XS GIS Cut Line= 3
      2449589.07     13586234.15      2450075.00     13586475.00
      2450474.95     13586375.01
#Sta/Elev= 30
  4458.1  301.32  4509.4  299.79  4543.6  296.94  4576.3  295.59  4650.5  290.54
  4879.9  276.78  4911.2  272.71  4919.2  268.91  4924.8  271.18  4941.6  266.84
  4947.2  267.94  4955.8  263.44  4964.0  261.10  4969.6  261.69  4978.1  259.56
  4992.0  254.03  4992.5  253.53  5003.3  254.03  5023.6  255.84  5031.4  258.96
  5059.7  267.02  5072.6  268.02  5113.8  268.66  5177.6  266.91  5258.1  270.82
  5307.1  275.85  5348.3  276.64  5381.8  280.61  5389.6  282.03  5412.7  281.40
#Mann=7,-1,0
  4458.1    0.07       0  4650.5    0.16       0  4919.2    0.12       0
  4992.0    0.07       0  5003.3    0.12       0  5177.6   0.035       0
  5381.8    0.05       0
Bank Sta=4992,5003.3
Exp/Cntr=0.3,0.1

Type RM Length L Ch R = 1,6976,455,455,455
BEGIN DESCRIPTION:
Stream0804 15.0
END DESCRIPTION:
XS GIS Cut Line= 3
      2449892.07     13587118.28      2450375.00     13586725.00
      2450474.99     13586525.02
#Sta/Elev= 30
  4381.7  282.89  4440.3  280.45  4450.0  279.43  4463.7  279.67  4471.7  278.85
  4515.2  277.38  4549.9  275.71  4620.3  270.90  4666.0  269.63  4698.6  268.59
  4855.1  267.11  4898.2  265.71  4912.6  264.70  4940.0  260.63  4947.8  258.70
  4968.6  257.42  4976.5  257.68  4983.0  255.22  4995.4  252.38  4995.9  251.88
  5006.6  251.88  5007.1  252.38  5018.5  253.10  5026.9  258.24  5040.9  262.70
  5085.6  264.80  5107.9  267.31  5138.7  269.38  5209.4  273.11  5228.1  274.58
#Mann=7,-1,0
  4381.7    0.07       0  4440.3    0.16       0  4515.2   0.035       0
  4666.0    0.16       0  4995.4    0.07       0  5007.1    0.16       0
  5209.4    0.05       0
Bank Sta=4995.4,5007.1
Exp/Cntr=0.3,0.1

Type RM Length L Ch R = 1,6521,476,476,476
BEGIN DESCRIPTION:
Stream0804 14.0
END DESCRIPTION:
XS GIS Cut Line= 3
      2450375.02     13587224.99      2450525.00     13587125.00
      2450674.97     13587025.02
#Sta/Elev= 30
  4815.7  263.92  4838.2  263.64  4859.2  263.84  4874.3  263.69  4893.4  263.83
  4923.8  263.81  4937.4  263.02  4959.9  258.69  4967.4  256.98  4973.4  254.24
  4976.6  251.35  4977.1  250.85  4987.8  250.85  4988.3  251.35  4993.0  252.85
  4999.0  252.85  5003.5  253.46  5009.5  253.74  5013.4  254.10  5045.5  256.65
  5054.5  258.06  5060.6  258.71  5068.1  259.80  5084.4  261.34  5096.6  262.86
  5126.7  264.98  5132.7  265.28  5147.7  265.58  5173.2  267.16  5176.2  267.16
#Mann=6,-1,0
  4815.7    0.07       0  4893.4    0.05       0  4976.6    0.05       0
  4988.3    0.05       0  5013.4    0.07       0  5084.4    0.05       0
Bank Sta=4976.6,4988.3
Exp/Cntr=0.3,0.1

Type RM Length L Ch R = 1,6045,441,441,441
BEGIN DESCRIPTION:
Stream0804 13.0
END DESCRIPTION:
XS GIS Cut Line= 3
      2450525.04     13587525.00      2450725.00     13587525.00
      2450875.04     13587525.00
#Sta/Elev= 30
  4804.6  258.84  4814.6  258.36  4834.6  258.02  4844.6  256.87  4854.6  256.37
  4864.6  256.58  4884.6  257.90  4904.6  257.62  4924.6  256.77  4944.6  255.06
  4964.6  254.40  4974.6  253.50  4984.6  249.37  4988.7  248.46  4989.2  247.96
  5000.0  247.96  5000.5  248.46  5002.1  250.26  5007.1  250.26  5014.6  253.45
  5024.6  255.56  5034.6  258.54  5044.6  261.03  5054.6  262.02  5064.6  262.49
  5084.6  262.92  5124.6  264.61  5144.6  264.81  5152.1  265.59  5154.6  265.59
#Mann=3,-1,0
  4804.6   0.035       0  4988.7   0.035       0  5000.5   0.035       0
Bank Sta=4988.7,5000.5
Exp/Cntr=0.3,0.1

Type RM Length L Ch R = 1,5604,460,460,460
BEGIN DESCRIPTION:
Stream0804 12.0
END DESCRIPTION:
XS GIS Cut Line= 3
      2450136.95     13587761.69      2450675.00     13587875.00
      2451131.59     13587642.13
#Sta/Elev= 30
  4444.1  265.95  4580.8  261.65  4738.5  259.94  4817.4  260.01  4861.1  260.60
  4869.4  259.60  4874.5  260.27  4881.5  260.03  4891.8  258.71  4902.0  255.93
  4912.2  252.31  4919.2  247.52  4924.4  251.86  4942.9  247.95  4953.1  246.84
  4968.3  246.81  4968.8  246.31  4980.1  246.81  5002.3  247.48  5007.9  250.04
  5016.4  251.47  5069.0  253.50  5113.4  258.89  5131.6  260.04  5180.1  262.40
  5230.2  263.23  5246.8  264.30  5402.4  269.25  5446.9  271.77  5506.5  277.14
#Mann=5,-1,0
  4444.1    0.05       0  4817.4    0.07       0  4968.3    0.07       0
  4980.1    0.07       0  5131.6    0.05       0
Bank Sta=4968.3,4980.1
Exp/Cntr=0.3,0.1

Type RM Length L Ch R = 1,5144,467,467,467
BEGIN DESCRIPTION:
Stream0804 11.0
END DESCRIPTION:
XS GIS Cut Line= 3
      2450374.96     13588074.99      2450775.00     13588175.00
      2451075.02     13588275.01
#Sta/Elev= 30
  4588.1  258.68  4670.6  258.68  4711.8  257.86  4735.0  257.93  4753.1  258.61
  4784.0  258.02  4907.7  258.93  4928.3  257.19  4936.0  255.92  4941.2  256.00
  4948.9  253.63  4969.5  251.87  4977.3  247.62  4982.4  249.80  4990.1  245.91
  4991.9  245.81  4992.4  245.31  5003.4  245.31  5003.9  245.81  5011.0  245.83
  5032.1  250.49  5074.2  251.98  5079.5  254.79  5084.8  256.71  5105.9  259.76
  5148.9  262.47  5221.8  267.73  5232.4  267.51  5264.0  270.09  5316.7  273.10
#Mann=4,-1,0
  4588.1    0.05       0  4991.9    0.07       0  5003.9    0.05       0
  5148.9    0.05       0
Bank Sta=4991.9,5003.9
Exp/Cntr=0.3,0.1

Type RM Length L Ch R = 1,4677,476,476,476
BEGIN DESCRIPTION:
Stream0804 10.0
END DESCRIPTION:
XS GIS Cut Line= 3
      2450325.02     13588325.01      2450725.00     13588625.00
      2450875.01     13588675.00
#Sta/Elev= 30
  4499.6  257.41  4649.6  256.37  4699.6  256.61  4721.5  256.00  4763.1  256.63
  4771.5  256.09  4806.9  256.59  4813.1  256.08  4849.6  255.64  4871.5  255.87
  4886.0  254.66  4899.6  252.45  4921.5  250.41  4956.9  248.00  4963.1  248.11
  4971.5  247.15  4977.7  247.55  4986.3  244.75  4986.8  244.25  4997.8  244.25
  4998.3  244.75  4999.6  245.60  5010.1  246.54  5020.7  248.50  5031.2  252.41
  5041.7  253.94  5074.3  260.51  5083.9  261.91  5153.8  265.57  5157.7  265.70
#Mann=5,-1,0
  4499.6    0.05       0  4986.3    0.05       0  4998.3    0.05       0
  5074.3    0.07       0  5153.8   0.035       0
Bank Sta=4986.3,4998.3
Exp/Cntr=0.3,0.1

Type RM Length L Ch R = 1,4201,455,455,455
BEGIN DESCRIPTION:
Stream0804 9.0
END DESCRIPTION:
XS GIS Cut Line= 3
      2450075.01     13588775.00      2450425.00     13588875.00
      2450724.99     13589025.00
#Sta/Elev= 30
  4636.3  255.62  4692.2  255.27  4719.5  253.89  4759.8  253.31  4804.0  249.94
  4823.5  251.59  4837.8  250.55  4844.3  251.45  4854.7  251.07  4871.6  244.51
  4876.8  244.20  4883.6  245.08  4905.4  249.56  4913.4  249.57  4917.1  250.26
  4927.5  250.09  4937.9  248.03  4949.6  243.02  4958.7  242.96  4963.0  241.84
  4963.5  241.34  4975.2  241.84  4983.4  244.74  5059.0  248.90  5098.1  254.43
  5142.8  254.69  5156.8  256.26  5170.8  259.01  5201.5  259.64  5335.7  259.56
#Mann=5,-1,0
  4636.3    0.05       0  4883.6    0.16       0  4913.4    0.05       0
  4963.0    0.05       0  4975.2    0.05       0
Bank Sta=4963,4975.2
Exp/Cntr=0.3,0.1

Type RM Length L Ch R = 1,3746,471,471,471
BEGIN DESCRIPTION:
Stream0804 8.0
END DESCRIPTION:
XS GIS Cut Line= 3
      2450025.02     13589125.01      2450275.00     13589275.00
      2450624.99     13589125.01
#Sta/Elev= 30
  4708.5  254.69  4751.6  254.16  4849.9  253.17  4873.0  252.80  4906.7  251.48
  4918.4  248.84  4928.1  245.04  4933.9  246.21  4949.5  243.25  4955.3  244.86
  4965.0  241.91  4991.0  238.64  4991.5  238.14  5002.7  238.14  5003.2  238.64
  5009.1  241.31  5021.8  242.56  5043.5  246.32  5067.1  247.17  5085.3  249.70
  5090.7  249.55  5097.9  250.52  5137.8  252.10  5214.0  252.06  5278.4  253.81
  5313.7  254.96  5337.3  256.81  5348.2  258.74  5359.1  259.53  5380.8  259.34
#Mann=7,-1,0
  4708.5    0.05       0  4751.6    0.16       0  4849.9    0.05       0
  4873.0    0.07       0  4991.0    0.07       0  5003.2    0.07       0
  5278.4    0.05       0
Bank Sta=4991,5003.2
Exp/Cntr=0.3,0.1

Type RM Length L Ch R = 1,3275,469,469,469
BEGIN DESCRIPTION:
Stream0804 7.0
END DESCRIPTION:
XS GIS Cut Line= 5
      2449518.24     13590090.81      2450301.39     13589798.61
      2450425.00     13589675.00      2450616.92     13589559.85
      2451315.94     13589335.33
#Sta/Elev= 30
  3989.3  283.77  4082.3  278.62  4278.5  271.75  4333.8  268.56  4505.0  262.29
  4560.3  261.45  4620.9  258.14  4651.2  257.85  4792.1  251.86  4943.4  248.94
  4956.2  247.32  4971.7  245.65  4985.8  242.71  4996.5  238.30  5000.0  238.30
  5001.6  237.07  5002.1  236.57  5014.0  237.07  5035.0  243.96  5071.9  248.99
  5223.7  250.83  5373.7  250.28  5482.0  251.57  5610.4  255.73  5653.0  258.69
  5704.9  260.13  5725.9  262.02  5799.5  265.62  5820.5  267.58  5958.0  274.76
#Mann=5,-1,0
  3989.3    0.05       0  4956.2   0.035       0  5001.6   0.035       0
  5014.0   0.035       0  5373.7    0.05       0
Bank Sta=5001.6,5014
Exp/Cntr=0.3,0.1

Type RM Length L Ch R = 1,2806,472,472,472
BEGIN DESCRIPTION:
Stream0804 6.0
END DESCRIPTION:
XS GIS Cut Line= 5
      2449700.19     13590140.44      2450571.91     13590061.73
      2450625.00     13590075.00      2450662.05     13590037.95
      2451370.58     13589567.29
#Sta/Elev= 30
  4075.4  276.51  4200.7  270.98  4281.0  268.59  4331.2  265.34  4391.5  263.78
  4562.2  255.57  4612.4  254.53  4692.7  250.80  4886.6  246.65  4913.6  246.09
  4933.7  243.22  4943.7  243.36  4954.8  242.15  4964.2  236.77  4974.5  235.69
  4988.9  235.68  4989.4  235.18  5001.3  235.68  5008.9  236.31  5019.5  244.43
  5033.7  248.08  5140.0  247.97  5301.3  247.15  5517.5  249.43  5755.3  259.50
  5776.3  262.28  5805.7  263.24  5848.5  267.26  5877.7  268.44  5908.4  271.17
#Mann=5,-1,0
  4075.4    0.05       0  4886.6     0.1       0  4988.9    0.05       0
  5001.3     0.1       0  5140.0    0.05       0
Bank Sta=4988.9,5001.3
Exp/Cntr=0.3,0.1

Type RM Length L Ch R = 1,2334,465,465,465
BEGIN DESCRIPTION:
Stream0804 5.0
END DESCRIPTION:
XS GIS Cut Line= 5
      2449904.26     13590658.80      2450499.25     13590468.94
      2450875.00     13590375.00      2450883.46     13590315.77
      2451470.22     13589666.38
#Sta/Elev= 30
  3996.1  277.71  4395.8  256.32  4605.7  247.75  4894.6  245.50  4902.3  244.97
  4915.2  239.84  4941.0  238.04  4948.7  235.08  4960.5  234.65  4961.0  234.15
  4973.0  234.65  4989.9  239.34  5010.5  238.52  5028.2  239.99  5058.5  245.61
  5120.4  245.50  5352.3  246.63  5614.6  250.54  5706.5  254.43  5763.3  258.70
  5777.5  257.63  5784.2  259.73  5805.9  261.93  5812.6  260.84  5841.0  262.48
  5883.6  266.54  5904.5  270.77  5918.7  269.82  5940.4  271.61  5943.0  273.09
#Mann=5,-1,0
  3996.1    0.05       0  4941.0     0.1       0  4960.5    0.05       0
  4973.0     0.1       0  5120.4    0.05       0
Bank Sta=4960.5,4973
Exp/Cntr=0.3,0.1

Type RM Length L Ch R = 1,1869,437,437,437
BEGIN DESCRIPTION:
Stream0804 4.0
END DESCRIPTION:
XS GIS Cut Line= 3
      2450425.03     13590874.99      2451225.00     13590625.00
      2451675.00     13589825.00
#Sta/Elev= 30
  4169.1  255.24  4268.9  250.66  4385.3  246.39  4455.6  244.45  4713.9  242.83
  4725.9  243.69  4745.3  243.04  4850.1  244.35  4888.3  243.42  4912.9  240.15
  4926.3  236.99  4944.4  236.00  4952.3  232.64  4952.8  232.14  4964.8  232.64
  4965.3  233.41  4991.0  237.20  5010.1  237.01  5030.2  242.80  5036.9  243.45
  5064.6  243.29  5096.1  240.25  5101.9  238.96  5119.2  240.69  5167.9  243.51
  5344.7  244.61  5366.4  247.55  5374.4  249.63  5409.8  254.12  5925.1  255.03
#Mann=7,-1,0
  4169.1    0.05       0  4268.9   0.035       0  4385.3    0.05       0
  4926.3    0.12       0  4952.3    0.07       0  4964.8    0.12       0
  5119.2    0.05       0
Bank Sta=4952.3,4964.8
Exp/Cntr=0.3,0.1

Type RM Length L Ch R = 1,1432,425,425,425
BEGIN DESCRIPTION:
Stream0804 3.0
END DESCRIPTION:
XS GIS Cut Line= 3
      2450374.96     13591625.03      2451575.00     13590725.00
      2452125.01     13590124.99
#Sta/Elev= 30
  3492.0  271.88  3496.5  271.93  3592.0  270.76  3855.6  252.54  4042.0  244.34
  4205.6  241.99  4684.8  240.73  4742.0  236.27  4778.5  235.97  4805.6  236.08
  4849.3  239.85  4889.8  239.27  4978.5  236.86  4992.0  234.60  4992.8  230.27
  4993.3  229.77  5005.4  230.27  5020.1  235.08  5070.1  237.65  5126.8  235.13
  5168.7  240.83  5268.7  242.38  5438.2  245.37  5452.4  245.18  5473.3  240.62
  5487.5  242.19  5496.1  240.90  5544.2  241.82  5601.0  248.87  5806.0  256.36
#Mann=7,-1,0
  3492.0    0.07       0  3496.5    0.05       0  4889.8    0.12       0
  4992.8    0.07       0  5005.4    0.12       0  5268.7    0.05       0
  5496.1    0.07       0
Bank Sta=4992.8,5005.4
Exp/Cntr=0.3,0.1
