--- Stream0834.prj (project) ---

Proj Title=Stream0834 Base Level Engineering
Current Plan=p01
Default Exp/Contr=0.3,0.1
English Units
Geom File=g01
Flow File=f01
Plan File=p01
Y Axis Title=Elevation
X Axis Title(PF)=Main Channel Distance
X Axis Title(XS)=Station
BEGIN DESCRIPTION:
Stream0834
END DESCRIPTION:
DSS Export Rating Curves= 0
DSS Export Rating Curve Sorted= 0
DSS Export Volume Flow Curves= 0
DXF OffsetX= 0
DXF OffsetY= 0
DXF ScaleX= 1
DXF ScaleY= 10

--- Stream0834.p01 (plan) ---

Plan Title=Multiple Run
Program Version=4.10
Short Identifier=Multiple
Geom File=g01
Flow File=f01
Subcritical Flow
K Sum by GR= 0
Std Step Tol= 0.01
Critical Tol= 0.01
Num of Std Step Trials= 20
Max Error Tol= 0.3
Flow Tol Ratio= 0.001
Split Flow NTrial= 30
Split Flow Tol= 0.02
Split Flow Ratio= 0.02
Log Output Level= 0
Friction Slope Method= 1
Unsteady Friction Slope Method= 2
Unsteady Bridges Friction Slope Method= 1
Parabolic Critical Depth
Global Vel Dist= 1 , 1 , 1
Global Log Level= 0
CheckData=True
Encroach Param=-1 ,0,0, 0
BEGIN DESCRIPTION:
Multiple Run
END DESCRIPTION:
Computation Interval=1HOUR
Output Interval=1HOUR
Run HTab= 0
Run UNet= 0
Run PostProcess= 0
Run WQNet= 0
UNET Theta= 1
UNET Theta Warmup= 1
UNET ZTol= 0.02
UNET ZSATol= 0.05
UNET MxIter= 20
UNET MaxInSteps= 0
UNET DtIC= 0
UNET DtMin= 0
UNET MaxCRTS= 20
UNET WFStab= 2
UNET SFStab= 1
UNET WFX= 1
UNET SFX= 1
UNET DSS MLevel= 4
UNET DZMax Abort= 100
UNET Convert EG Bridges= 0
UNET Use Existing IB Tables=-1
UNET Froude Reduction=False
UNET Froude Limit= 1
UNET Froude Power= 10
UNET Time Slicing=0,0, 5
UNET Junction Losses=0
Instantaneous Interval=1HOUR
Write IC File= 0
Write IC File at Sim End=0
Echo Input=False
Echo Parameters=False
Echo Output=False
Write Detailed= 0
WQ AD Non Conservative
WQ ULTIMATE=-1
WQ Max Comp Step=1HOUR
WQ Output Interval=15MIN
WQ Output Selected Increments= 0
WQ Output face flow=0
WQ Output face velocity=0
WQ Output face area=0
WQ Output face dispersion=0
WQ Output cell volume=0
WQ Output cell surface area=0
WQ Output cell continuity=0
WQ Output cumulative cell continuity=0
WQ Output face conc=0
WQ Output face dconc_dx=0
WQ Output face courant=0
WQ Output face peclet=0
WQ Output face adv mass=0
WQ Output face disp mass=0
WQ Output cell mass=0
WQ Output cell source sink temp=0
WQ Output cell source sink nsm=0
WQ Output MaxMinRange=-1
WQ Daily Max Min Mean=-1
WQ Daily Range=0
WQ Daily Time=0
WQ Create Restart=0
WQ Fixed Restart=0
WQ System Summary=0
WQ Use Fixed Temperature=0
Sorting and Armoring Iterations= 10
XS Update Threshold= 0.02
Hydraulics Update Threshold= 0.02
Energy Slope Method= 1
Volume Change Method= 0
XS Weighting Method= 0
Number of US Weighted Cross Sections= 1
Number of DS Weighted Cross Sections= 1
Upstream XS Weight=0.25
Main XS Weight=0.5
Downstream XS Weight=0.25
Number of DS XS's Weighted with US Boundary= 1
Upstream Boundary Weight= 1
Weight of XSs Associated with US Boundary= 0
Number of US XS's Weighted with DS Boundary= 1
Downstream Boundary Weight= 0.5
Weight of XSs Associated with DS Boundary= 0.5
Sediment Output Level= 4
Mass or Volume Output= 0
Output Increment Type= 1
Profile and TS Output Increment= 10
XS Output Flag= 0
XS Output Increment= 10
Disregard all LS=0
Disregard all Conn=0
Disregard all Breaches=0
Disregard all Pumps=0

--- Stream0834.f01 (steady flow) ---

Flow Title=Multiple
Number of Profiles=7
Profile Names=10-year,25-year,50-year,1pct_min,100-year,1pct_plu,500-year
River Rch & RM= Stream0834,Reach-1,29710
     773    1267    1722    1133    2261    4512    3864
River Rch & RM= Stream0834,Reach-1,28694
    1067    1773    2429    1610    3212    6408    5563
River Rch & RM= Stream0834,Reach-1,21878
    1808    3062    4247    2842    5671   11316   10028
River Rch & RM= Stream0834,Reach-1,12193
    2863    4927    6909    4667    9311   18578   16773
River Rch & RM= Stream0834,Reach-1,8654
    3092    5339    7503    5080   10135   20222   18338
River Rch & RM= Stream0834,Reach-1,6694
    3082    5296    7417    5002    9980   19912   17918
River Rch & RM= Stream0834,Reach-1,578
    3031    5197    7269    4895    9767   19488   17486
Boundary for River Rch & Prof#=Stream0834,Reach-1,1
Up Type=0
Dn Type=3
Dn Slope=0.005
Boundary for River Rch & Prof#=Stream0834,Reach-1,2
Up Type=0
Dn Type=3
Dn Slope=0.005
Boundary for River Rch & Prof#=Stream0834,Reach-1,3
Up Type=0
Dn Type=3
Dn Slope=0.005
Boundary for River Rch & Prof#=Stream0834,Reach-1,4
Up Type=0
Dn Type=3
Dn Slope=0.005
Boundary for River Rch & Prof#=Stream0834,Reach-1,5
Up Type=0
Dn Type=3
Dn Slope=0.005
Boundary for River Rch & Prof#=Stream0834,Reach-1,6
Up Type=0
Dn Type=3
Dn Slope=0.005
Boundary for River Rch & Prof#=Stream0834,Reach-1,7
Up Type=0
Dn Type=3
Dn Slope=0.005

--- Stream0834.g01 (geometry) ---

Geom Title=Existing Conditions
Program Version=4.10

River Reach=Stream0834      ,Reach-1
Reach XY= 30
        2476375.       13569125.      2477019.55     13569372.53
      2478164.82     13572114.68      2479035.68     13572524.25
      2480119.07     13572477.24      2480390.36     13572775.11
      2480615.31     13572335.18      2480914.59     13572375.99
      2481266.84     13572768.95      2481172.94     13573869.15
      2480828.08     13574223.34      2481669.17      13574572.7
       2482024.3      13575385.7      2482034.41     13576531.62
      2482723.04     13576830.89      2482488.34     13577338.31
      2482769.14     13577472.95      2483064.36     13577175.55
      2483669.17      13577572.7      2483980.83      13579727.3
      2485822.95     13581830.84      2485377.05     13582430.86
       2485378.1     13583273.82      2486017.25     13583218.45
      2486072.33     13584269.71      2486571.67     13583882.59
      2486817.25     13584068.55      2487082.81     13584831.19
      2487871.47     13585626.46        2487725.       13586525.

Type RM Length L Ch R = 1 ,29710   ,558,558,558
BEGIN DESCRIPTION:
Stream0834 51.0
END DESCRIPTION:
XS GIS Cut Line= 3
      2475842.03     13569368.49      2476353.59     13569190.69
      2476777.74     13568875.69
#Sta/Elev= 30
    4397  283.25  4409.1  283.03  4569.5  282.31  4605.6  278.67  4622.5  281.85
  4637.2  287.26  4643.6   288.1  4654.2  287.19    4663  284.91  4668.3  280.84
  4675.4  277.81  4682.9  277.04  4694.1   276.4  4707.2  278.87  4730.5  279.52
  4834.2   279.2  4844.4  280.18  4849.7  278.47  4875.5   279.7  4880.8  277.76
  4887.1  277.31  4965.2  273.99  5022.4  274.79  5041.3  273.47  5041.5  272.97
  5045.3  273.47  5101.7  275.74  5164.5  280.31  5463.9  284.47  5466.9  284.47
#Mann= 6 ,-1 , 0
    4397     .12       0  4409.1     .07       0  4682.9     .12       0
  5041.3     .05       0  5045.3     .12       0  5463.9     .07       0
Bank Sta=5041.3,5045.3
XS Rating Curve= 0 ,0
Exp/Cntr=0.3,0.1

Type RM Length L Ch R = 1 ,29152   ,458,458,458
BEGIN DESCRIPTION:
Stream0834 50.0
END DESCRIPTION:
XS GIS Cut Line= 3
      2476425.02     13569824.97        2476925.       13569275.
        2477075.       13569125.
#Sta/Elev= 30
  4260.9  289.87  4353.1  286.24  4374.1  286.19  4388.2  283.11  4409.5  284.17
  4423.4  282.14    4445  283.47  4465.9  281.66  4544.3  278.49  4662.3  276.04
  4671.4  275.26  4678.8  273.29  4706.8  268.54  4756.5  270.17  4777.5  269.77
  4784.9  267.74  4789.7  267.53  4789.9  267.03  4793.7  267.53  4813.3  276.21
  4883.6  275.53  4919.4  271.28  4961.9  271.03  4976.1  269.63  4982.9  270.73
  5002.9  271.79  5018.3  272.93  5046.6  276.82  5109.3  278.91  5216.3  283.08
#Mann= 6 ,-1 , 0
  4260.9     .05       0  4662.3     .12       0  4789.7     .05       0
  4793.7     .12       0  5002.9     .07       0  5109.3     .12       0
Bank Sta=4789.7,4793.7
XS Rating Curve= 0 ,0
Exp/Cntr=0.3,0.1

Type RM Length L Ch R = 1 ,28694   ,442,442,442
BEGIN DESCRIPTION:
Stream0834 49.0
END DESCRIPTION:
XS GIS Cut Line= 3
      2476674.98     13570025.01        2477075.       13569675.
      2477325.01     13569474.99
#Sta/Elev= 30
  4468.5  286.66  4512.5  285.06  4532.6   283.9  4546.8  284.48  4567.7  282.56
  4574.8  280.69  4596.2  279.68  4610.4  279.77  4624.7  280.73  4638.9  279.53
  4704.1  277.04  4745.2   275.5  4837.3  273.81  4929.3  273.55  4944.6   271.8
  4964.4  268.57  4986.3  266.45  5013.6  266.51  5019.6  263.05  5019.9  262.55
  5023.4  262.55  5023.6  263.05    5028   263.6    5036   268.2  5056.9  270.35
  5071.3  273.02  5141.7  275.73  5149.7  276.52  5205.7  277.13  5320.2  280.71
#Mann= 6 ,-1 , 0
  4468.5     .05       0  4512.5     .12       0  4704.1     .05       0
  4944.6     .12       0  5019.6     .05       0  5023.6     .12       0
Bank Sta=5019.6,5023.6
XS Rating Curve= 0 ,0
Exp/Cntr=0.3,0.1

Type RM Length L Ch R = 1 ,28252   ,447,447,447
BEGIN DESCRIPTION:
Stream0834 48.0
END DESCRIPTION:
XS GIS Cut Line= 3
      2476924.96     13570125.01        2477325.       13570025.
      2477524.99       13569975.
#Sta/Elev= 30
  4591.5  277.55  4609.6  277.73  4622.5  276.31  4641.5  276.22  4743.6  272.77
  4838.9  270.65    4857  269.51  4862.1  269.78  4914.5  265.92  4931.7  265.05
  4972.9  265.03  4980.7  264.29  4985.8   262.3  4991.5  260.94  4991.8  260.44
  4995.3  260.44  4995.5  260.94  5001.3  262.88  5006.4  262.88  5014.2  264.36
  5021.9  264.42  5055.4  268.94  5068.3  271.08    5076  273.26  5096.6  274.09
  5104.4  275.35  5109.5  274.68  5117.2  275.39  5151.3   276.3    5210  278.45
#Mann= 7 ,-1 , 0
  4591.5     .12       0  4641.5    .035       0  4743.6     .05       0
  4914.5     .12       0  4991.5     .05       0  4995.5     .12       0
  5151.3     .07       0
Bank Sta=4991.5,4995.5
XS Rating Curve= 0 ,0
Exp/Cntr=0.3,0.1

Type RM Length L Ch R = 1 ,27805   ,415,415,415
BEGIN DESCRIPTION:
Stream0834 47.0
END DESCRIPTION:
XS GIS Cut Line= 3
      2476925.03       13570375.        2477325.       13570375.
      2477675.04     13570224.98
#Sta/Elev= 30
  4600.4  280.48  4641.4  278.35  4710.4  275.33  4739.7  275.47  4770.4  271.95
  4780.4   271.7  4800.4  274.26  4810.4  273.63  4830.4  269.34  4838.1  269.23
  4850.4  269.85  4880.4  268.38  4930.4  262.87  4938.3  260.56  4938.6  260.06
  4942.1  260.06  4942.4  260.56  4950.4  260.59  4970.4  262.81  4980.4  263.32
  5008.9  262.87    5062  262.98  5109.2   264.9  5130.9  268.22  5138.2  270.34
  5167.2  271.61  5196.2   274.6  5272.4  279.33  5297.1  279.87  5381.2  282.95
#Mann= 8 ,-1 , 0
  4600.4     .12       0  4641.4     .05       0  4739.7     .12       0
  4838.1    .035       0  4938.3    .035       0  4942.4    .035       0
  5008.9     .07       0  5297.1     .05       0
Bank Sta=4938.3,4942.4
XS Rating Curve= 0 ,0
Exp/Cntr=0.3,0.1

Type RM Length L Ch R = 1 ,27390   ,455,455,455
BEGIN DESCRIPTION:
Stream0834 46.0
END DESCRIPTION:
XS GIS Cut Line= 3
      2476874.97     13570474.99        2477425.       13570625.
        2477775.       13570325.
#Sta/Elev= 30
    4419  282.34  4527.1  277.31  4587.8  274.67  4719.6  270.69  4736.4  269.31
  4761.1  267.98  4778.4   271.7  4792.2  271.46  4802.5  270.16  4812.9  266.91
  4823.3   265.9  4897.6  266.03  4947.7  259.18  4971.8  259.31  4978.8  260.55
  4986.5  267.23  5023.8   265.6  5039.1  262.77  5045.6  259.06  5068.9   256.4
  5107.3  255.64  5107.5  255.14  5111.4  255.64  5145.5  257.41  5156.6  259.79
  5215.4  268.53  5272.8  274.23  5279.4  276.79  5289.3  277.15  5450.1  284.45
#Mann= 11 ,-1 , 0
    4419     .05       0  4527.1     .12       0  4587.8     .05       0
  4736.4     .12       0  5023.8    .035       0  5068.9     .12       0
  5107.3     .05       0  5111.4     .12       0  5156.6     .07       0
  5215.4     .12       0  5289.3     .05       0
Bank Sta=5107.3,5111.4
XS Rating Curve= 0 ,0
Exp/Cntr=0.3,0.1

Type RM Length L Ch R = 1 ,26935   ,432,432,432
BEGIN DESCRIPTION:
Stream0834 45.0
END DESCRIPTION:
XS GIS Cut Line= 3
      2476874.99       13571425.        2477675.       13570975.
      2477975.01     13570574.99
#Sta/Elev= 30
  4086.5  279.25  4109.5  278.18  4121.9  279.43  4137.8  277.66  4189.8  275.42
  4202.8  276.81  4218.8  275.06  4327.5  271.07  4343.1  272.71    4359  270.86
  4380.7  270.34  4672.7  265.63  4688.5  265.64  4710.2  263.72  4731.9  266.83
  4740.5  266.37  4747.8  262.92  4828.3  261.32  4850.4   260.9  4937.1  262.64
    4947  261.78    4967  255.71  4967.2  255.21  4971.1  255.71  4981.4  258.44
  4993.4  258.84  5127.8  264.92  5248.4  269.79  5450.5  280.18  5504.4   281.5
#Mann= 9 ,-1 , 0
  4086.5     .05       0  4672.7     .07       0  4828.3     .05       0
    4967     .05       0  4971.1     .05       0  4993.4     .05       0
  5127.8     .07       0  5248.4     .05       0  5450.5    .035       0
Bank Sta=4967,4971.1
XS Rating Curve= 0 ,0
Exp/Cntr=0.3,0.1

Type RM Length L Ch R = 1 ,26503   ,440,440,440
BEGIN DESCRIPTION:
Stream0834 44.0
END DESCRIPTION:
XS GIS Cut Line= 3
      2476975.02       13571425.        2477775.       13571375.
        2478075.       13571075.
#Sta/Elev= 30
  4194.2  276.84  4214.2   275.5  4234.3  276.35  4304.4  273.06  4324.4  271.29
  4334.5  272.36  4444.7  267.14  4592.5  263.74  4702.5  262.79  4715.2  262.15
  4725.2  260.49  4735.2  260.91  4752.8  263.84  4765.3  264.28  4775.3  261.87
  4795.3  259.54  4835.4  261.45  4918.1  259.29  4943.5  253.85  4943.8  253.35
  4947.7  253.85  4955.7  256.02  4965.7  257.18  4988.4  257.44  5016.2  256.95
  5052.3  256.86  5080.6  259.72    5138  260.54  5193.7  260.88    5420  270.61
#Mann= 7 ,-1 , 0
  4194.2     .05       0  4702.5     .07       0  4943.5     .05       0
  4947.7     .07       0  4988.4     .05       0  5016.2     .07       0
    5138     .05       0
Bank Sta=4943.5,4947.7
XS Rating Curve= 0 ,0
Exp/Cntr=0.3,0.1

Type RM Length L Ch R = 1 ,26063   ,488,488,488
BEGIN DESCRIPTION:
Stream0834 43.0
END DESCRIPTION:
XS GIS Cut Line= 3
      2477625.01     13572474.97        2478075.       13571675.
        2478275.       13571425.
#Sta/Elev= 30
  4081.7  276.65  4116.6  274.57  4221.7  269.36  4228.2   269.1    4333  264.59
  4444.3     261  4537.7  260.51  4559.4  258.11    4575  259.48  4581.1  261.68
  4586.8  262.13    4597  261.73  4602.8  259.27  4618.7  256.87  4666.9  257.67
  4780.6  257.79    4862  254.65  4889.4  254.46  4964.2  254.97  4976.6   254.5
  4989.1   252.5  4989.5     252  4994.1   252.5  4996.7  253.94  5009.5   254.1
  5056.5  256.74  5099.6  259.59  5124.3  259.87  5285.1  264.67  5319.7  266.68
#Mann= 15 ,-1 , 0
  4081.7     .07       0  4116.6     .05       0  4221.7     .07       0
  4228.2     .05       0    4333    .035       0  4444.3     .12       0
  4666.9     .05       0    4862     .07       0  4889.4     .05       0
  4989.1     .05       0  4994.1     .05       0  5009.5     .07       0
  5056.5     .05       0  5124.3    .035       0  5285.1     .05       0
Bank Sta=4989.1,4994.1
XS Rating Curve= 0 ,0
Exp/Cntr=0.3,0.1

Type RM Length L Ch R = 1 ,25575   ,445,445,445
BEGIN DESCRIPTION:
Stream0834 42.0
END DESCRIPTION:
XS GIS Cut Line= 3
      2477775.03     13572524.97        2478175.       13572125.
      2478624.97     13571525.04
#Sta/Elev= 30
  4430.5  273.63  4738.8  260.39  4769.9  258.16  4799.4  260.34  4812.3  260.15
  4840.6  255.67  4854.7  256.66    4882  256.16  4925.4  256.06  4934.9  254.45
  4967.9  250.67  4979.5  247.89  4979.9  247.39  4984.5  247.89  4992.6  253.52
    4999  253.52    5118  252.08  5146.1  254.39  5332.6  256.62  5346.1  257.97
  5359.7  257.26  5453.4  259.84  5488.9   262.6  5503.4  262.45  5544.7  264.95
  5559.7   266.9  5596.1  266.62  5638.9  268.84  5703.4   273.8  5746.1  274.44
#Mann= 9 ,-1 , 0
  4430.5     .05       0  4738.8     .07       0  4799.4     .12       0
    4882     .07       0  4934.9     .05       0  4979.5     .05       0
  4984.5     .05       0    4999     .07       0  5544.7     .05       0
Bank Sta=4979.5,4984.5
XS Rating Curve= 0 ,0
Exp/Cntr=0.3,0.1

Type RM Length L Ch R = 1 ,25130   ,476,476,476
BEGIN DESCRIPTION:
Stream0834 41.0
END DESCRIPTION:
XS GIS Cut Line= 3
      2477774.98     13572675.01        2478575.       13572275.
      2478774.99     13571625.02
#Sta/Elev= 30
  4111.6  276.01  4152.9  274.34  4304.5   268.8    4447     262  4528.1  260.18
  4582.6  257.03  4595.2  259.35  4617.5  259.72  4648.3  254.53  4656.7  255.77
  4751.7  255.34  4774.1   257.1  4796.4  254.74  4841.1  253.74  4894.2  250.63
  4961.3  250.79  4969.7  249.63  4972.8  246.49  4973.2  245.99  4977.8  246.49
  4997.7  250.75  5027.6  251.11  5055.1  252.65  5173.5  254.77  5309.5   254.2
  5397.7  256.23  5501.1  261.34  5631.8  270.78  5675.3  272.07  5686.1  272.26
#Mann= 6 ,-1 , 0
  4111.6     .07       0  4152.9     .05       0  4582.6     .07       0
  4972.8     .05       0  4977.8     .07       0  5675.3     .05       0
Bank Sta=4972.8,4977.8
XS Rating Curve= 0 ,0
Exp/Cntr=0.3,0.1

Type RM Length L Ch R = 1 ,24654   ,451,451,451
BEGIN DESCRIPTION:
Stream0834 40.0
END DESCRIPTION:
XS GIS Cut Line= 3
      2478375.01     13573274.99        2478975.       13572475.
        2478825.     13571675.03
#Sta/Elev= 30
  4004.8  268.26  4210.8  265.23  4402.8  259.14  4459.1  258.14  4512.1  254.78
  4526.7  256.35  4562.1  256.23  4576.7  254.26  4658.5  252.84  4741.2  251.76
  4782.9  250.35  4791.2  248.81  4832.9  249.22  4841.2  251.08  4854.8  251.51
  4912.1  251.27  4954.8  248.13  4976.7  248.23  4988.7  246.43  4989.1  245.93
  4993.8  246.43  4997.5  248.88  5001.7  249.42  5036.2  247.99  5088.7  250.93
    5198     252    5483  253.44  5645.8  260.27  5776.9  268.38  5818.7  270.73
#Mann= 9 ,-1 , 0
  4004.8     .05       0  4210.8     .07       0  4402.8     .05       0
  4459.1     .07       0  4658.5     .05       0  4988.7     .05       0
  4993.8     .05       0    5198     .07       0  5776.9     .05       0
Bank Sta=4988.7,4993.8
XS Rating Curve= 0 ,0
Exp/Cntr=0.3,0.1

Type RM Length L Ch R = 1 ,24203   ,498,498,498
BEGIN DESCRIPTION:
Stream0834 39.0
END DESCRIPTION:
XS GIS Cut Line= 3
      2478925.03     13572974.96        2479375.       13572425.
      2478874.99     13571624.99
#Sta/Elev= 30
  4289.3  255.31  4408.3  254.58  4503.5  253.72  4540.8  253.12  4566.3  253.92
  4629.5  253.02  4694.1   252.3  4807.5  248.44  4850.6  249.76  4900.1  248.64
  4922.4  246.92  4935.3  247.84  4949.6  247.38  4957.5   244.1  4961.3  243.63
  4961.7  243.13  4966.7  243.63  4971.9   245.4  4978.4  244.62  4992.7  246.68
  5013.4   247.3  5035.3  249.59  5188.6  250.98  5379.1  250.66  5494.6   250.8
  5624.9  255.86  5669.6  258.48  5719.2  260.63  5848.9   269.5  5943.3  272.53
#Mann= 9 ,-1 , 0
  4289.3     .05       0  4408.3     .07       0  4503.5     .05       0
  4540.8     .07       0  4629.5     .05       0  4961.3     .05       0
  4966.7     .05       0  5379.1     .07       0  5669.6     .05       0
Bank Sta=4961.3,4966.7
XS Rating Curve= 0 ,0
Exp/Cntr=0.3,0.1

Type RM Length L Ch R = 1 ,23705   ,639,639,639
BEGIN DESCRIPTION:
Stream0834 38.0
END DESCRIPTION:
XS GIS Cut Line= 3
      2479225.02     13573224.98        2479875.       13572425.
      2479054.81     13571574.49
#Sta/Elev= 30
  3973.6  257.62    4024  256.95  4148.1  254.44  4272.3  251.95  4463.4  247.47
  4541.7   247.7  4570.5  246.71    4592  244.29  4656.5  244.95  4712.7  246.88
  4770.2  246.29  4781.8  242.41  4782.3  241.91  4787.3  242.41  4798.2  246.05
  4805.4  247.25  4848.5  245.63  4977.1  245.87  5027.6  246.48  5223.7  248.69
  5440.3  247.47  5440.8  247.44  5471.1  246.37  5513.6  246.41  5793.2  249.61
  5830.7  250.51  5994.4   257.3  6121.7  260.63  6143.1   260.2  6185.9  261.37
#Mann= 12 ,-1 , 0
  3973.6    .035       0    4024     .05       0  4148.1     .07       0
  4272.3     .05       0  4781.8    .035       0  4787.3     .05       0
  4977.1    .035       0  5027.6     .05       0  5440.3     .07       0
  5440.8     .05       0  5793.2     .07       0  5830.7     .05       0
Bank Sta=4781.8,4787.3
XS Rating Curve= 0 ,0
Exp/Cntr=0.3,0.1

Type RM Length L Ch R = 1 ,23066   ,1188,1188,1188
BEGIN DESCRIPTION:
Stream0834 37.0
END DESCRIPTION:
XS GIS Cut Line= 3
      2479774.97     13573475.04      2480287.77     13572908.33
      2480769.74      13571305.5
#Sta/Elev= 30
  4059.3  254.88  4490.9  247.32  4936.1  247.46  4962.8   244.6  4974.4  240.06
  4994.1  237.42  5007.4  241.73    5015  242.12  5223.9  242.04  5265.6   243.6
    5282  242.39    5297  237.65  5328.3  239.02  5345.3  236.41  5345.7  235.91
  5350.9  236.41  5359.6  238.25  5380.5  238.09  5386.3  240.82  5391.6  239.16
  5452.4  242.18  5594.9  240.14  5620.7  237.67  5672.9  242.68  5860.8  245.89
  6063.7  253.56  6088.7  254.84    6292  264.56  6444.6   265.4  6497.3  265.46
#Mann= 6 ,-1 , 0
  4059.3     .05       0  5345.3     .05       0  5350.9     .05       0
  6063.7     .07       0  6088.7     .05       0  6444.6    .035       0
Bank Sta=5345.3,5350.9
XS Rating Curve= 0 ,0
Exp/Cntr=0.3,0.1

Type RM Length L Ch R = 1 ,21878   ,443,443,443
BEGIN DESCRIPTION:
Stream0834 36.0
END DESCRIPTION:
XS GIS Cut Line= 3
      2479875.01     13573624.99        2481075.       13572525.
      2481874.96     13572075.02
#Sta/Elev= 30
  3372.1  255.81  3548.7  250.44  3867.5  244.69  3966.8  245.52  4101.2  249.51
    4186  248.21  4355.9  241.77  4412.6  240.66  4589.6  241.32  4632.1  240.12
  4667.3  241.34  4709.8  240.01  4773.4  240.42  4844.3     238  4936.1  238.85
  4971.9  237.31    5002  237.71  5008.7  234.49  5009.2  233.99  5018.7  234.49
  5029.6   234.6  5045.5  239.19  5072.9   241.6  5096.3  241.91  5191.5   242.2
  5240.9  244.47  5418.4  243.68  5542.7  246.48  5807.3  255.45  5917.8  261.33
#Mann= 5 ,-1 , 0
  3372.1     .05       0    5002     .07       0  5008.7     .05       0
  5018.7     .07       0  5096.3     .05       0
Bank Sta=5008.7,5018.7
XS Rating Curve= 0 ,0
Exp/Cntr=0.3,0.1

Type RM Length L Ch R = 1 ,21435   ,477,477,477
BEGIN DESCRIPTION:
Stream0834 35.0
END DESCRIPTION:
XS GIS Cut Line= 3
      2480125.02     13573574.99        2481325.       13572875.
      2481724.99     13572475.01
#Sta/Elev= 30
  3614.9  248.07  3761.7  244.16  3900.6  241.69    4104  243.78  4199.9  240.63
  4221.4   240.8  4309.5  238.59  4477.8  238.62  4499.3  239.27    4515  238.33
    4558  238.06  4573.7  237.03  4579.5  238.13  4595.2  235.95  4659.7  234.77
  4691.1  235.79  4894.6  237.28  4953.3  236.32    4981  237.47  4996.3  236.64
  5001.2  234.21  5013.1  233.98  5013.6  233.48  5023.5  233.98  5032.4  234.05
  5046.5  238.54  5074.8  239.62  5272.8  240.76  5400.1  243.79  5569.8  252.39
#Mann= 3 ,-1 , 0
  3614.9     .05       0  5013.1     .05       0  5023.5     .05       0
Bank Sta=5013.1,5023.5
XS Rating Curve= 0 ,0
Exp/Cntr=0.3,0.1

Type RM Length L Ch R = 1 ,20958   ,465,465,465
BEGIN DESCRIPTION:
Stream0834 34.0
END DESCRIPTION:
XS GIS Cut Line= 3
      2480325.04     13573924.97        2481125.       13573275.
      2481925.04     13572874.98
#Sta/Elev= 30
  3969.2  247.98    4125  244.38  4211.2  240.55    4403  235.66    4459  236.98
  4594.8  236.58  4637.9  237.49    4652  237.68  4673.1  236.21  4692.5  236.48
  4716.2  237.42  4850.5  238.15  4879.3  235.48  4885.7  232.92  4902.8  229.08
  4903.3  228.58  4913.3  229.08  4914.4  233.33  4922.4  234.39  4935.5  233.92
    4964  235.51  4992.7  235.95  5029.2  238.24  5097.8  237.34  5215.2  238.14
  5290.6  236.39  5380.1  237.12  5438.8  239.86  5656.8  243.73  5894.4  252.28
#Mann= 6 ,-1 , 0
  3969.2     .05       0  4637.9    .035       0  4692.5     .05       0
  4902.8    .035       0  4913.3     .05       0  5029.2     .05       0
Bank Sta=4902.8,4913.3
XS Rating Curve= 0 ,0
Exp/Cntr=0.3,0.1

Type RM Length L Ch R = 1 ,20493   ,916,916,916
BEGIN DESCRIPTION:
Stream0834 33.0
END DESCRIPTION:
XS GIS Cut Line= 3
      2480375.04     13573974.99        2481175.       13573675.
      2481975.03     13573074.98
#Sta/Elev= 30
  4145.6  247.27  4276.4  243.98  4423.2  238.34  4572.8  235.05  4594.1  233.22
  4618.1  232.74  4636.8  232.51    4668  234.83  4722.3  235.82  4753.4  233.85
  4775.7  233.54  4954.6   234.8  4978.6  233.78  4979.6  229.47  4980.1  228.97
  4990.1  229.47  5007.3  229.56  5028.1  231.83  5036.4  237.08  5071.8  238.81
    5150  236.22  5227.3  236.41  5271.8  236.42  5336.4  234.62  5442.7  235.45
  5521.8  234.93  5742.7  240.34  5887.6  245.45  5968.1  248.95    6000  250.75
#Mann= 6 ,-1 , 0
  4145.6     .05       0  4979.6    .035       0  4990.1     .05       0
  5227.3     .05       0  5887.6     .07       0  5968.1     .05       0
Bank Sta=4979.6,4990.1
XS Rating Curve= 0 ,0
Exp/Cntr=0.3,0.1

Type RM Length L Ch R = 1 ,19577   ,438,438,438
BEGIN DESCRIPTION:
Stream0834 32.0
END DESCRIPTION:
XS GIS Cut Line= 3
      2480574.99       13574575.        2480975.       13574325.
      2482075.01     13573124.99
#Sta/Elev= 30
  4513.2  251.82  4641.9  246.15  4645.3  246.01  4694.2  244.21  4709.6  241.02
  4730.8  244.19  4767.3  240.79  4890.6  236.87  4913.6  234.45  4919.5  230.52
  4925.9   229.4  4961.9  230.94  4965.9  228.91  4966.4  228.41  4976.7  228.91
  4977.2  230.61    4992  231.41  5055.5  230.57  5183.2  235.52  5664.1  233.49
  5770.8  234.97    5891  233.37  6077.5  234.26  6147.6  236.46  6201.4  237.64
  6296.1  240.28    6372   244.5  6499.1  247.92  6607.2  252.06  6612.8  252.18
#Mann= 11 ,-1 , 0
  4513.2     .05       0  4641.9    .035       0  4645.3     .05       0
  4965.9     .05       0  4976.7     .05       0  6077.5     .07       0
  6147.6     .05       0  6201.4     .07       0  6296.1     .05       0
  6499.1     .07       0  6607.2     .05       0
Bank Sta=4965.9,4976.7
XS Rating Curve= 0 ,0
Exp/Cntr=0.3,0.1

Type RM Length L Ch R = 1 ,19139   ,425,425,425
BEGIN DESCRIPTION:
Stream0834 31.0
END DESCRIPTION:
XS GIS Cut Line= 3
      2480625.03     13574824.98        2481375.       13574375.
      2482175.01     13573574.99
#Sta/Elev= 30
  4125.4  253.19  4443.7   238.9  4475.2  236.66  4488.8  240.57  4498.6  240.53
  4510.2   238.8  4519.9  235.43  4533.5  234.65  4547.1  235.37  4671.4  233.56
  4780.4  234.97  4887.1  233.59    4965  230.67  4976.7  225.51  4986.8  224.39
  4987.3  223.89  4997.7  224.39    5000  227.96  5016.1  230.62  5049.3  232.58
  5268.7  231.75    5372  230.01  5410.1  229.16    5495  231.76  5590.9  232.99
  5735.4   236.3  5820.3  236.43  5913.1   239.6  5975.8  241.53  6131.4  249.71
#Mann= 11 ,-1 , 0
  4125.4     .05       0  4443.7    .035       0  4671.4     .12       0
  4887.1     .05       0  4986.8     .05       0  4997.7     .05       0
  5016.1     .07       0  5049.3     .05       0    5372     .12       0
  5590.9     .05       0  5913.1     .07       0
Bank Sta=4986.8,4997.7
XS Rating Curve= 0 ,0
Exp/Cntr=0.3,0.1

Type RM Length L Ch R = 1 ,18714   ,470,470,470
BEGIN DESCRIPTION:
Stream0834 30.0
END DESCRIPTION:
XS GIS Cut Line= 3
      2480475.03     13574924.99        2481675.       13574625.
      2482474.97     13574225.01
#Sta/Elev= 30
  3758.5  259.33    4029  248.42  4350.7  232.77  4376.9  237.21  4387.2  237.26
  4400.1  236.74  4418.2   231.2  4449.1  232.39  4520.9  232.11  4572.8  232.47
  4634.6  235.07  4714.8  233.23  4923.2  231.03  5003.8  228.77  5084.8  230.85
  5115.6  229.62  5272.1  229.88  5330.8  227.52  5333.6  223.15  5334.1  222.65
  5344.7  223.15  5367.1  229.93  5389.5  234.04  5404.8  235.46  5423.1  236.73
  5473.4  238.68  5568.4  239.89  5695.1   245.3  5876.1  253.37  5889.8  253.79
#Mann= 10 ,-1 , 0
  3758.5     .05       0  4350.7    .035       0  4520.9     .12       0
  4714.8     .05       0  5333.6     .05       0  5344.7     .05       0
  5404.8     .12       0  5423.1     .05       0  5695.1     .07       0
  5876.1     .05       0
Bank Sta=5333.6,5344.7
XS Rating Curve= 0 ,0
Exp/Cntr=0.3,0.1

Type RM Length L Ch R = 1 ,18244   ,453,453,453
BEGIN DESCRIPTION:
Stream0834 29.0
END DESCRIPTION:
XS GIS Cut Line= 3
      2480675.02       13575025.        2481875.       13575025.
      2482675.03     13574274.98
#Sta/Elev= 30
  3804.3  250.91  4094.3  237.64  4356.4  230.56  4386.9  230.04  4424.3  229.03
  4434.3  229.73  4454.3  234.91  4474.3  235.36  4490.3  231.03  4514.3  227.85
  4554.3  231.05    4681     233  4684.3  233.02  4754.3   232.7  4764.3  231.12
  4774.3   227.4  4778.7  222.65  4779.2  222.15  4789.8  222.65  4804.3  227.25
  4814.3   227.4  5149.8  228.04  5236.7  230.01  5296.8  232.18  5392.8  234.91
  5605.8  240.93  5852.6  251.06  5902.8  254.48  5970.2  255.79  6100.9  259.79
#Mann= 14 ,-1 , 0
  3804.3     .05       0  4356.4     .12       0  4386.9     .05       0
  4490.3     .12       0    4681    .035       0  4684.3     .05       0
  4778.7     .05       0  4789.8     .05       0  5149.8     .07       0
  5236.7     .05       0  5296.8     .07       0  5392.8     .05       0
  5852.6     .07       0  5970.2     .05       0
Bank Sta=4778.7,4789.8
XS Rating Curve= 0 ,0
Exp/Cntr=0.3,0.1

Type RM Length L Ch R = 1 ,17791   ,453,453,453
BEGIN DESCRIPTION:
Stream0834 28.0
END DESCRIPTION:
XS GIS Cut Line= 3
      2480825.04     13575225.01        2482025.       13575425.
      2482424.99     13575075.01
#Sta/Elev= 30
  3787.2  243.83  4202.8  228.95  4344.7  227.99  4577.9  230.87  4598.2  228.96
  4618.5  229.55  4628.6  232.53  4648.9  233.94  4666.6  232.26  4671.7  233.47
  4689.4  229.73  4709.7  228.44  4727.5  229.79  4828.2  228.21  4906.8  225.18
  5017.5  225.82  5083.1  221.16  5083.6  220.66  5094.2  221.16  5117.1  223.91
    5138  223.78  5159.8  227.45    5195  228.44  5209.2  227.66  5223.4  224.11
  5258.6  222.45  5289.8  232.15  5294.6  234.35  5375.8  235.53  5535.2   240.2
#Mann= 7 ,-1 , 0
  3787.2     .05       0  4828.2    .035       0  4906.8     .05       0
  5083.1     .05       0  5094.2     .05       0  5289.8     .07       0
  5375.8     .05       0
Bank Sta=5083.1,5094.2
XS Rating Curve= 0 ,0
Exp/Cntr=0.3,0.1

Type RM Length L Ch R = 1 ,17338   ,487,487,487
BEGIN DESCRIPTION:
Stream0834 27.0
END DESCRIPTION:
XS GIS Cut Line= 3
      2480674.97     13575274.99        2481875.       13575775.
      2482674.97     13575475.01
#Sta/Elev= 30
  3700.4   248.9    4247  228.99  4376.2  227.59  4805.1  228.25  4845.6  228.48
  4924.6  226.83  4932.7  223.17  4938.1  223.55    4951  219.64  4956.6   217.8
    4962  219.05  4962.3  217.36  4962.8  216.86  4973.5  217.36  4985.8   220.5
  5021.8  223.56  5107.2  226.01  5131.3  224.71  5139.3  225.39  5156.2  231.14
  5162.9  231.23  5181.1  230.35  5192.7   224.6  5203.3  223.49  5216.7  226.67
  5269.1  227.22  5587.6  232.06  5716.8  234.43  5819.5  236.35  5854.8  237.53
#Mann= 13 ,-1 , 0
  3700.4     .05       0    4247     .07       0  4376.2     .05       0
  4805.1     .12       0  4845.6    .035       0    4951     .12       0
  4962.3     .05       0  4973.5     .12       0  5162.9     .07       0
  5269.1     .05       0  5587.6     .07       0  5716.8     .05       0
  5819.5     .07       0
Bank Sta=4962.3,4973.5
XS Rating Curve= 0 ,0
Exp/Cntr=0.3,0.1

Type RM Length L Ch R = 1 ,16851   ,419,419,419
BEGIN DESCRIPTION:
Stream0834 26.0
END DESCRIPTION:
XS GIS Cut Line= 3
      2480775.02       13576425.        2481975.       13576225.
      2482774.96     13575525.03
#Sta/Elev= 30
  3778.7  246.46  3805.8  245.07  4083.8  232.88  4325.2  226.21  4569.4  224.94
  4750.8   227.5    4833  224.79  4934.4  223.89  4954.7  222.06  4967.4  215.09
    4979  214.97  4987.1  214.88  4987.6  214.38  4998.3  214.88  5016.6  218.17
  5023.2  221.71  5065.9  220.29  5122.9  225.44  5349.7  226.02    5364  224.61
  5378.2  227.81  5384.8  230.58  5392.4  230.88  5406.7  229.89  5413.3  227.63
  5427.6  225.71  5441.8  227.78  5757.3  234.21  5971.3  237.43  6058.2  239.31
#Mann= 10 ,-1 , 0
  3778.7     .05       0  3805.8    .035       0  4083.8     .05       0
  4325.2    .035       0  4750.8     .12       0    4979     .05       0
  4987.1     .05       0  4998.3     .05       0  5757.3     .07       0
  5971.3     .05       0
Bank Sta=4987.1,4998.3
XS Rating Curve= 0 ,0
Exp/Cntr=0.3,0.1

Type RM Length L Ch R = 1 ,16432   ,939,939,939
BEGIN DESCRIPTION:
Stream0834 25.0
END DESCRIPTION:
XS GIS Cut Line= 3
        2480825.       13576525.        2482025.       13576525.
      2482825.01     13575774.99
#Sta/Elev= 30
  3781.4  245.82  3818.7  244.43  3940.2  239.53  4191.4  228.72  4324.8  225.52
  4480.6  225.04  4611.4  226.51  4693.4  225.41  4881.4  224.87  4939.6  221.28
  4995.3  219.43  4997.1  215.87  4997.6  215.37  5008.3  215.87    5031  219.53
    5052  219.99  5073.5  224.26  5105.2  224.56    5174  224.23  5367.7   224.3
  5412.8  224.91  5497.9  226.37  5526.3  225.12  5554.6  230.92  5568.8  230.36
  5582.9  226.21  5632.3  228.98    5967   233.9  5982.4  234.55    6078  235.66
#Mann= 15 ,-1 , 0
  3781.4     .05       0  3818.7    .035       0  3940.2     .05       0
  4324.8    .035       0  4480.6     .07       0  4693.4    .035       0
  4939.6     .05       0  4997.1     .05       0  5008.3     .05       0
  5105.2    .035       0    5174     .05       0  5367.7     .07       0
  5412.8     .05       0    5967     .07       0  5982.4     .05       0
Bank Sta=4997.1,5008.3
XS Rating Curve= 0 ,0
Exp/Cntr=0.3,0.1

Type RM Length L Ch R = 1 ,15493   ,777,777,777
BEGIN DESCRIPTION:
Stream0834 24.0
END DESCRIPTION:
XS GIS Cut Line= 3
      2481125.02       13576625.        2482725.       13576875.
      2482974.96     13576675.03
#Sta/Elev= 30
  3379.5  235.31  3476.1  230.22  3500.1  229.57    3535  228.16  3647.5  225.23
  3827.3  224.71  3930.6  226.72  3993.3  224.79  4085.6  224.22  4199.3   223.9
  4280.3  222.69  4460.8  222.18  4659.3   221.9  4735.7  222.15  4766.1   221.5
  4786.3  220.19  4826.8  219.94  4847.1  218.85  4938.2   218.7  4996.4  217.68
  5020.5  218.03  5057.3  215.72  5057.8  215.22  5068.1  215.22  5068.6  215.72
  5070.1  217.62  5076.5  218.46  5084.5  221.53  5248.9  223.89    5319  225.57
#Mann= 11 ,-1 , 0
  3379.5     .05       0  3500.1    .035       0    3535     .05       0
  3647.5    .035       0  3827.3     .07       0  4085.6     .05       0
  4460.8     .12       0  4659.3    .035       0  5057.3    .035       0
  5068.6    .035       0  5248.9     .05       0
Bank Sta=5057.3,5068.6
XS Rating Curve= 0 ,0
Exp/Cntr=0.3,0.1

Type RM Length L Ch R = 1 ,14716   ,1440,1440,1440
BEGIN DESCRIPTION:
Stream0834 23.0
END DESCRIPTION:
XS GIS Cut Line= 3
      2482271.67     13577728.09      2482596.76     13577548.73
      2483213.26     13576674.42
#Sta/Elev= 30
  4538.8  219.65  4631.1  218.84  4726.1   217.7  4815.5  218.15  4839.6  217.81
  4873.8  215.16  4926.9  214.07  4939.2  213.19  4946.5  210.72  4948.1  209.59
  4948.6  209.09  4959.8  209.59  4962.6  213.71  4968.7  214.28  5064.7  216.79
  5182.9  216.74  5227.4  217.09  5263.1  216.05  5298.8  217.14  5334.5  215.69
  5378.9  218.77  5405.9  216.85  5463.6  219.34  5622.7   222.4  5649.7  224.01
  5735.9  225.08  5807.9   227.8  5851.7  227.31  5887.9  229.29  5979.9  231.69
#Mann= 10 ,-1 , 0
  4538.8    .035       0  4631.1     .05       0  4815.5    .035       0
  4946.5     .12       0  4948.1     .05       0  4959.8     .12       0
  5064.7     .05       0  5182.9     .12       0  5463.6    .035       0
  5887.9     .05       0
Bank Sta=4948.1,4959.8
XS Rating Curve= 0 ,0
Exp/Cntr=0.3,0.1

Type RM Length L Ch R = 1 ,13276   ,1083,1083,1083
BEGIN DESCRIPTION:
Stream0834 21.0
END DESCRIPTION:
XS GIS Cut Line= 4
      2482383.77     13577784.11      2483314.12     13577828.95
      2483728.84     13577571.15      2483616.76     13576820.21
#Sta/Elev= 30
  3643.1  218.95  3949.1  216.91  3976.8  217.44  4094.9   215.1    4235   217.1
  4403.1  216.19  4455.3  217.78    4554  216.96  4823.7  217.35  4881.7  213.06
  4970.2  211.08    4976  209.85  4979.6  206.48  4980.1  205.98  4991.4  206.48
  4999.5  209.74  5012.7  210.23  5034.8  217.65  5043.4   218.2  5123.7  216.83
  5139.8  218.36  5200.5  218.12  5240.9  224.86  5257.2  223.59  5262.2  224.86
  5291.5  221.34  5383.9  226.47  5487.3  230.13  5507.6  231.11  5822.1  240.97
#Mann= 10 ,-1 , 0
  3643.1    .035       0  3949.1     .07       0  3976.8    .035       0
  4403.1     .12       0    4554    .035       0  4979.6    .035       0
  4991.4    .035       0  5383.9     .05       0  5487.3     .07       0
  5507.6     .05       0
Bank Sta=4979.6,4991.4
XS Rating Curve= 0 ,0
Exp/Cntr=0.3,0.1

Type RM Length L Ch R = 1 ,12193   ,781,781,781
BEGIN DESCRIPTION:
Stream0834 19.0
END DESCRIPTION:
XS GIS Cut Line= 3
      2482475.02     13579674.98      2483740.05     13578557.51
      2485522.26     13577358.16
#Sta/Elev= 30
  3329.1  236.19  3894.3  220.97  3908.6  220.37  4038.5  218.44  4177.8  214.78
  4866.2  213.62  4985.5  209.63  5029.7  206.29  5037.3  199.12  5037.8  198.62
  5052.1  199.12  5053.3  199.22  5080.7  206.89  5109.5  205.98  5122.7  203.07
  5137.7  207.48  5152.7  202.92  5173.7  209.54  5230.4  210.82  5338.7  214.87
  5673.9  215.85  5794.4  214.68  5836.5  221.99  5866.5  215.27  5923.5  220.86
  6069.5  223.15  6076.4   223.2  6392.4  230.21  6817.3  239.81  7165.2  242.32
#Mann= 15 ,-1 , 0
  3329.1     .05       0  3894.3    .035       0  3908.6     .05       0
  4038.5     .12       0  4177.8     .05       0  4985.5     .12       0
  5037.3     .05       0  5052.1     .12       0  5053.3     .05       0
  5109.5     .12       0  5230.4    .035       0  5673.9     .05       0
  6069.5    .035       0  6076.4     .07       0  6392.4     .05       0
Bank Sta=5037.3,5052.1
XS Rating Curve= 0 ,0
Exp/Cntr=0.3,0.1

Type RM Length L Ch R = 1 ,11412   ,488,488,488
BEGIN DESCRIPTION:
Stream0834 17.0
END DESCRIPTION:
XS GIS Cut Line= 3
      2482675.03     13580424.97        2483875.       13579225.
      2485674.97     13578025.02
#Sta/Elev= 30
  3302.7  260.94  3310.6   260.9  3366.6  258.22  3642.1  247.63  3741.1  240.78
  4278.5  215.82    4599  210.74  4721.8  210.28  4738.6  210.21  4858.3  206.91
  4971.4  207.26  5002.7  202.41    5004   198.5  5004.5     198  5022.5   198.5
  5028.3  202.88  5079.3     208  5316.7  210.11  5475.9  205.38  5540.5  212.68
    5694  212.95    6161  215.14    6176  216.25  6189.5  221.91  6197.1  222.48
  6212.1  221.25  6231.6  216.01  6254.1  218.48  6441.9  223.39    7163  239.49
#Mann= 9 ,-1 , 0
  3302.7     .05       0  3310.6     .07       0  3366.6     .05       0
    4599    .035       0  4721.8     .07       0  4738.6    .035       0
    5004    .035       0  5022.5    .035       0    5694     .05       0
Bank Sta=5004,5022.5
XS Rating Curve= 0 ,0
Exp/Cntr=0.3,0.1

Type RM Length L Ch R = 1 ,10924   ,461,461,461
BEGIN DESCRIPTION:
Stream0834 16.0
END DESCRIPTION:
XS GIS Cut Line= 3
      2483375.03     13580274.97        2483975.       13579675.
      2485174.97     13578675.02
#Sta/Elev= 30
  4156.6  231.87  4312.1  225.46  4393.4  220.46  4467.7  215.18  4583.4  213.42
  4664.5  211.94  4799.1  210.04  4906.1  209.69  4934.4  207.84  4962.7  199.88
  4967.5  197.19    4968  196.69  4986.1  197.19  4990.9   204.6  5001.6  205.85
  5069.5  203.81  5125.5  208.15  5168.5   208.1  5217.9  212.34  5442.3  210.69
  5495.2  209.81  6027.6  212.07  6299.4  216.42  6389.5  217.92  6403.7   216.8
  6410.9  217.03  6432.4  223.08    6461  217.99  6475.4   219.5  6567.1  221.26
#Mann= 10 ,-1 , 0
  4156.6     .12       0  4393.4     .05       0  4583.4     .12       0
  4664.5     .05       0  4799.1    .035       0  4967.5    .035       0
  4986.1    .035       0  5442.3     .05       0  6299.4     .12       0
  6403.7     .05       0
Bank Sta=4967.5,4986.1
XS Rating Curve= 0 ,0
Exp/Cntr=0.3,0.1

Type RM Length L Ch R = 1 ,10463   ,445,445,445
BEGIN DESCRIPTION:
Stream0834 15.0
END DESCRIPTION:
XS GIS Cut Line= 3
      2483674.96     13580325.02        2484275.       13579975.
      2485474.98     13578775.02
#Sta/Elev= 30
  4300.4  221.22  4431.5  215.32  4564.6  213.49  4591.9  212.09  4785.8  208.31
  4826.8  206.27  4842.5   207.1  4885.5  203.96  4930.7  204.24  4971.9  203.51
  4981.4  198.75  4982.9  196.47  4983.4  195.97  5001.5  196.47  5023.4  209.05
  5027.3   209.3  5079.9  210.82  5249.6  209.09    5589  209.73  5716.3  213.24
  6041.6  212.24  6154.7  213.49  6365.5  218.48  6409.3  218.84  6423.4  223.48
  6437.6  223.36  6451.7  220.99  6465.8  220.63  6539.1  223.71  6692.1  229.11
#Mann= 8 ,-1 , 0
  4300.4      .1       0  4785.8    .035       0  4930.7     .12       0
  4982.9     .05       0  5001.5     .12       0  5027.3     .05       0
  6365.5     .12       0  6539.1     .05       0
Bank Sta=4982.9,5001.5
XS Rating Curve= 0 ,0
Exp/Cntr=0.3,0.1

Type RM Length L Ch R = 1 ,10018   ,444,444,444
BEGIN DESCRIPTION:
Stream0834 14.0
END DESCRIPTION:
XS GIS Cut Line= 3
      2484124.98     13580675.01        2484575.       13580275.
      2485775.03     13579074.97
#Sta/Elev= 30
  4397.9  220.93  4770.3  212.91  4835.5  211.18    4914   206.4  4929.3   206.2
    4936  202.72  4962.6  196.83  4963.1  196.33  4981.3  196.83  4996.7  201.75
  5042.4  207.05  5103.1  208.73  5141.4  209.42  5226.3  206.64  5311.1  208.69
  5466.7  207.47    5594   208.9  5698.4  208.18    5732  207.96  5827.7  208.11
  5856.8  208.03  6117.2  209.87  6329.4  216.49  6463.8  222.45  6499.1  223.33
  6513.2  225.75  6527.4   224.3  6555.6  226.93  6625.8   228.8  6697.1  231.46
#Mann= 13 ,-1 , 0
  4397.9     .05       0  4770.3     .12       0  4835.5    .035       0
    4914     .12       0  4962.6     .05       0  4981.3     .12       0
  5103.1     .05       0  5698.4    .035       0    5732     .05       0
  5827.7    .035       0  5856.8     .05       0  6463.8     .07       0
  6625.8     .05       0
Bank Sta=4962.6,4981.3
XS Rating Curve= 0 ,0
Exp/Cntr=0.3,0.1

Type RM Length L Ch R = 1 ,9574    ,466,466,466
BEGIN DESCRIPTION:
Stream0834 13.0
END DESCRIPTION:
XS GIS Cut Line= 3
      2483675.03     13581174.98        2484875.       13580575.
      2486075.03     13579374.97
#Sta/Elev= 30
  3658.4  235.19  3733.3  233.05    4181  218.18    4209  218.71  4292.8   215.9
  4485.7  212.75  4642.2  208.05  4874.2  205.99  4910.6  205.45  4955.3   201.3
  4977.6   198.4  4987.9   193.6  4988.4   193.1  5006.6   193.6  5014.1  197.37
  5048.8  203.94  5070.7  207.38  5113.1  206.95  5184.3  209.19  5367.7  205.86
  5608.1  207.58  6046.5  206.47  6244.5  209.19  6386.1  213.22    6399  213.56
  6566.2   219.3  6626.3  222.17  6637.9  225.03  6668.8  224.17  6697.1  225.28
#Mann= 11 ,-1 , 0
  3658.4    .035       0  3733.3     .05       0  4874.2      .1       0
  4987.9     .05       0  5006.6      .1       0  5048.8    .035       0
  5184.3     .05       0  6386.1    .035       0    6399     .05       0
  6566.2    .035       0  6637.9     .05       0
Bank Sta=4987.9,5006.6
XS Rating Curve= 0 ,0
Exp/Cntr=0.3,0.1

Type RM Length L Ch R = 1 ,9108    ,454,454,454
BEGIN DESCRIPTION:
Stream0834 12.0
END DESCRIPTION:
XS GIS Cut Line= 3
      2483925.02       13581125.        2485125.       13580925.
      2486325.01     13579724.99
#Sta/Elev= 30
    3783  226.46  3965.5  220.13  3998.4  220.28  4054.2     217    4115  215.44
  4654.8  206.29  4776.5  206.55  4903.8  201.62  4971.6  201.37  4989.4   198.5
    4997  195.76  5003.1  195.76  5004.3  194.19  5004.8  193.69    5023  194.19
  5027.8  194.38    5042     200  5084.4  204.09  5098.5  207.28  5126.8  205.74
    5241  206.24  5289.3  206.24  5429.3   205.1  5519.8  204.92  5579.4  204.95
  5607.6  206.64  5655.3  205.03  6215.8  208.71  6385.5  212.98  6696.6  224.18
#Mann= 9 ,-1 , 0
    3783     .05       0  4903.8      .1       0  5004.3     .05       0
    5023      .1       0    5241     .07       0  5289.3      .1       0
  5429.3     .07       0  5519.8    .035       0  5655.3     .05       0
Bank Sta=5004.3,5023
XS Rating Curve= 0 ,0
Exp/Cntr=0.3,0.1

Type RM Length L Ch R = 1 ,8654    ,948,948,948
BEGIN DESCRIPTION:
Stream0834 11.0
END DESCRIPTION:
XS GIS Cut Line= 3
      2484074.97       13581425.        2485275.       13581325.
      2486475.01       13581325.
#Sta/Elev= 30
  3791.7  222.25  3929.7  220.06  4082.7  215.65  4203.2  213.83  4233.3  212.01
  4273.4  212.26  4484.1  207.77  4614.6  203.14  4855.4   205.4  4925.6  205.32
  4954.3  204.01  4998.4  199.31  5016.5  193.61    5017  193.11  5035.2  193.61
  5065.9  199.83  5155.9     201  5215.9   203.9  5385.9  201.53  5415.9  198.94
  5425.9  195.13  5445.9  199.67  5465.9   202.3  5523.3  202.32  5621.7  202.43
  5755.9  205.01  5905.9   210.3  6122.1  224.06  6166.5   226.3  6195.9   227.7
#Mann= 9 ,-1 , 0
  3791.7     .12       0  3929.7     .05       0  4954.3      .1       0
  5016.5     .05       0  5035.2      .1       0  5523.3     .12       0
  5621.7     .05       0  6122.1    .035       0  6166.5     .05       0
Bank Sta=5016.5,5035.2
XS Rating Curve= 0 ,0
Exp/Cntr=0.3,0.1

Type RM Length L Ch R = 1 ,7706    ,1012,1012,1012
BEGIN DESCRIPTION:
Stream0834 9.0
END DESCRIPTION:
XS GIS Cut Line= 3
      2484024.97       13581675.        2485825.       13581975.
      2486425.04     13581724.98
#Sta/Elev= 30
  3174.7  224.06  4149.8  200.72  4180.9  198.98  4208.8  194.26  4236.7  198.58
  4330.5  201.97  4411.6  202.98  4461.9  200.35  4601.6  202.98  4715.1  201.65
  4857.6  197.61  4910.8  199.77  4938.7  197.24  4979.3   198.3  5004.2   193.2
  5004.7   192.7  5024.1   193.2  5032.1  199.55    5038  201.27  5144.2  199.62
  5221.1  202.22  5278.1  214.68  5292.1  217.08  5309.6  216.44  5345.7   213.8
  5385.9  217.01    5428  214.48  5433.4  212.15  5457.3  211.99  5649.6  220.38
#Mann= 9 ,-1 , 0
  3174.7     .05       0  4149.8     .07       0  4461.9    .035       0
  4715.1     .12       0  5004.2     .05       0  5024.1     .12       0
  5278.1     .07       0  5309.6     .12       0  5385.9     .05       0
Bank Sta=5004.2,5024.1
XS Rating Curve= 0 ,0
Exp/Cntr=0.3,0.1

Type RM Length L Ch R = 1 ,6694    ,1342,1342,1342
BEGIN DESCRIPTION:
Stream0834 8.0
END DESCRIPTION:
XS GIS Cut Line= 3
      2483874.97       13582475.        2485475.       13582725.
      2487025.02     13581574.98
#Sta/Elev= 30
  3385.2  229.83  3390.2  229.71  3510.5  224.53  3987.3     209  4417.6  210.12
  4626.5  203.62  4840.2   188.2  4845.2  193.15  4919.5  192.57    4954  191.84
  4965.7  184.55  4966.2  184.05  4985.8  184.55  5026.6  196.91  5149.5  201.76
  5244.8   199.9  5312.4  188.44  5347.9  193.08  5354.1  189.26  5362.5  194.59
  5368.7  189.69    5398  198.47  5521.5  199.83  5620.8  198.19  5642.5  198.98
  5719.4  202.79  5851.5  208.82  5984.3  217.62  6470.4  216.29  6934.7  223.27
#Mann= 15 ,-1 , 0
  3385.2     .07       0  3390.2     .12       0  3510.5    .035       0
  3987.3     .05       0  4626.5    .035       0  4919.5     .12       0
  4965.7     .05       0  4985.8     .12       0  5149.5      .1       0
  5244.8     .12       0  5521.5      .1       0  5620.8     .07       0
  5642.5     .12       0  5719.4     .07       0  5851.5     .05       0
Bank Sta=4965.7,4985.8
XS Rating Curve= 0 ,0
Exp/Cntr=0.3,0.1

Type RM Length L Ch R = 1 ,5352    ,882,882,882
BEGIN DESCRIPTION:
Stream0834 6.0
END DESCRIPTION:
XS GIS Cut Line= 3
        2485025.       13584075.      2486015.41      13583175.5
      2486575.84      13582121.9
#Sta/Elev= 30
  3689.4   222.3  3880.3   208.9    4079  199.39  4323.8  198.33    4475  195.42
  4539.2  197.02  4742.5   194.5  4871.6  189.89  4878.4  188.01  4885.8  189.86
  4928.4  188.14  4935.2  185.71  4942.6  185.98  4946.6  179.88  4947.1  179.38
  4966.9  179.88  4977.7  189.45  4991.9  193.34  5035.3   196.5  5073.5  196.24
  5093.9   196.5  5183.5  195.82  5293.4  196.79  5315.1  197.64  5536.4  204.36
  5623.3  206.08  5825.7  212.03  5913.6  212.31  5951.9  215.07  6220.7  215.13
#Mann= 12 ,-1 , 0
  3689.4     .12       0  4323.8     .05       0  4742.5      .1       0
  4946.6     .05       0  4966.9      .1       0  5073.5     .07       0
  5093.9    .035       0  5183.5     .07       0  5293.4     .12       0
  5315.1     .07       0  5536.4     .12       0  5623.3     .05       0
Bank Sta=4946.6,4966.9
XS Rating Curve= 0 ,0
Exp/Cntr=0.3,0.1

Type RM Length L Ch R = 1 ,4470    ,1648,1648,1648
BEGIN DESCRIPTION:
Stream0834 4.0
END DESCRIPTION:
XS GIS Cut Line= 3
      2485175.04     13584624.97        2485975.       13583975.
        2487525.       13582375.
#Sta/Elev= 30
  3969.4  237.86    4098  232.58    4432  206.57  4537.5  200.98  4645.7   198.1
  4815.5  191.31  4943.8  191.15  4986.5  190.05  5134.5     192  5198.1  198.66
  5304.3  196.83  5391.8  192.37  5445.7  187.87  5463.6  178.54  5464.1  178.04
    5484  178.54    5488  186.24  5495.2  188.95  5542.7  190.41    5587     195
  6007.6  197.34  6089.6  198.42  6380.9  203.56  6577.1  206.69  6605.4  207.83
  6612.6  210.14  6852.9  212.15  6881.2  215.08  6981.9  216.55  7227.8  219.25
#Mann= 11 ,-1 , 0
  3969.4     .12       0  4645.7     .07       0  4943.8     .12       0
  5391.8      .1       0  5463.6     .05       0    5484      .1       0
  5542.7     .12       0  6007.6    .035       0  6089.6     .12       0
  6380.9     .07       0  6981.9     .05       0
Bank Sta=5463.6,5484
XS Rating Curve= 0 ,0
Exp/Cntr=0.3,0.1
